--- Bear Creek 2.prj (project) ---

Proj Title=Bear Creek 2 Base Level Engineering
Current Plan=p01
Default Exp/Contr=0.3,0.1
English Units
Geom File=g01
Flow File=f01
Plan File=p01
Y Axis Title=Elevation
X Axis Title(PF)=Main Channel Distance
X Axis Title(XS)=Station
BEGIN DESCRIPTION:
Bear Creek 2
END DESCRIPTION:
DSS Export Rating Curves= 0
DSS Export Rating Curve Sorted= 0
DSS Export Volume Flow Curves= 0
DXF OffsetX= 0
DXF OffsetY= 0
DXF ScaleX= 1
DXF ScaleY= 10

--- Bear Creek 2.p01 (plan) ---

Plan Title=Multiple Run
Short Identifier=Multiple
Geom File=g01
Flow File=f01
Subcritical Flow
K Sum by GR= 0
Std Step Tol= 0.01
Critical Tol= 0.01
Num of Std Step Trials= 20
Max Error Tol= 0.3
Flow Tol Ratio= 0.001
Split Flow NTrial= 30
Split Flow Tol= 0.02
Split Flow Ratio= 0.02
Log Output Level= 0
Friction Slope Method= 1
Unsteady Friction Slope Method= 2
Unsteady Bridges Friction Slope Method= 1
Parabolic Critical Depth
Global Vel Dist=  1 , 1 , 1
Global Log Level= 0
CheckData=True
Encroach Param= -1, 0, 0, 0
BEGIN DESCRIPTION:
Multiple Run
END DESCRIPTION:

--- Bear Creek 2.f01 (steady flow) ---

Flow Title=Multiple
Number of Profiles=7
Profile Names=10-year,25-year,50-year,1pct_min,100-year,1pct_plu,500-year
River Rch & RM= Bear Creek 2,Reach-1,71356
     258     398     519     328     655    1306    1026
River Rch & RM= Bear Creek 2,Reach-1,70473
    1199    2062    2886    1950    3891    7763    6995
River Rch & RM= Bear Creek 2,Reach-1,66779
    1607    2792    3934    2671    5330   10634    9684
River Rch & RM= Bear Creek 2,Reach-1,59154
    2662    4738    6785    4673    9325   18605   17444
River Rch & RM= Bear Creek 2,Reach-1,53183
    3718    6717    9715    6753   13474   26884   25672
River Rch & RM= Bear Creek 2,Reach-1,51801
    4584    8348   12141    8481   16921   33762   32560
River Rch & RM= Bear Creek 2,Reach-1,48935
    5566   10180   14847   10392   20736   41373   40062
River Rch & RM= Bear Creek 2,Reach-1,42825
    6015   11026   16105   11288   22523   44939   43630
River Rch & RM= Bear Creek 2,Reach-1,40110
    6283   11531   16855   11821   23587   47062   45749
River Rch & RM= Bear Creek 2,Reach-1,38964
    6604   12120   17719   12425   24792   49467   48073
River Rch & RM= Bear Creek 2,Reach-1,34671
    6619   12141   17741   12434   24810   49502   48055
River Rch & RM= Bear Creek 2,Reach-1,31382
    7331   13483   19740   13858   27651   55170   53730
River Rch & RM= Bear Creek 2,Reach-1,24754
    7526   13849   20283   14244   28421   56707   55260
River Rch & RM= Bear Creek 2,Reach-1,21175
    9945   18400   27057   19071   38051   75923   74474
River Rch & RM= Bear Creek 2,Reach-1,16009
   10377   19205   28247   19911   39727   79266   77761
River Rch & RM= Bear Creek 2,Reach-1,8296
   10481   19392   28515   20093   40092   79993   78425
River Rch & RM= Bear Creek 2,Reach-1,5036
   10587   19587   28802   20296   40495   80799   79210
Boundary for River Rch & Prof#=Bear Creek 2,Reach-1,1
Up Type=0
Dn Type=3
Dn Slope=0.005
Boundary for River Rch & Prof#=Bear Creek 2,Reach-1,2
Up Type=0
Dn Type=3
Dn Slope=0.005
Boundary for River Rch & Prof#=Bear Creek 2,Reach-1,3
Up Type=0
Dn Type=3
Dn Slope=0.005
Boundary for River Rch & Prof#=Bear Creek 2,Reach-1,4
Up Type=0
Dn Type=3
Dn Slope=0.005
Boundary for River Rch & Prof#=Bear Creek 2,Reach-1,5
Up Type=0
Dn Type=3
Dn Slope=0.005
Boundary for River Rch & Prof#=Bear Creek 2,Reach-1,6
Up Type=0
Dn Type=3
Dn Slope=0.005
Boundary for River Rch & Prof#=Bear Creek 2,Reach-1,7
Up Type=0
Dn Type=3
Dn Slope=0.005

--- Bear Creek 2.g01 (geometry) ---

Geom Title=Existing Conditions
Program Version=4.10

River Reach=Bear Creek 2    ,Reach-1
Reach XY= 30
        1799275.       13970175.      1801921.45     13968123.53
      1802176.05     13963185.44      1803283.14     13959768.96
      1804838.57     13959061.53       1805551.3     13957798.18
      1808118.54     13955732.74        1810125.       13955225.
       1810325.4       13954050.      1809725.52     13951559.78
      1809880.73     13950822.45      1811876.25     13949378.45
      1813305.38     13949495.47      1815091.65     13946257.47
      1817219.53     13945127.45      1816954.79      13943144.5
      1819228.31     13942933.02        1821125.       13944225.
      1822573.72     13944121.48      1823366.86     13943431.06
      1824833.15     13940928.37       1826554.9     13941325.09
        1828675.       13940675.      1829067.44       13939575.
        1828315.     13937436.24      1830554.83      13937925.3
      1832071.42     13936982.89       1833223.5     13937121.54
      1834680.56     13934630.62        1837725.       13933425.

Type RM Length L Ch R = 1 ,71356   ,417,417,417
BEGIN DESCRIPTION:
Bear Creek 2 135.0
END DESCRIPTION:
XS GIS Cut Line= 3
        1799975.     13970675.01        1799575.       13970075.
      1798975.03     13969475.03
#Sta/Elev= 30
  4279.1 2273.72  4282.1 2273.72  4286.6 2273.53  4307.7  2273.1  4415.8 2270.51
  4430.8 2270.06    4539 2267.27  4617.1 2265.38  4662.2 2264.44  4725.3 2262.75
  4812.4 2260.59  4848.5 2259.89  4920.6 2258.79  4986.7 2258.11  5012.4 2258.03
  5012.6 2257.53  5016.1 2257.53  5016.4 2258.03  5056.8 2258.26  5155.8 2259.91
  5382.1 2265.06  5389.1 2265.09  5396.2 2265.38  5481.1  2267.2  5551.8 2269.24
  5763.9 2276.24  5806.3 2277.84  5834.6 2278.69  5845.2 2279.11  5848.7 2279.11
#Mann= 3 ,-1 , 0
  4279.1     .07       0  5012.4     .05       0  5016.4     .07       0
Bank Sta=5012.4,5016.4
XS Rating Curve= 0 ,0
Exp/Cntr=0.3,0.1

Type RM Length L Ch R = 1 ,70939   ,466,466,466
BEGIN DESCRIPTION:
Bear Creek 2 134.0
END DESCRIPTION:
XS GIS Cut Line= 3
      1800074.99     13970374.99        1799825.       13969775.
      1799225.01     13969275.01
#Sta/Elev= 30
  4344.7 2268.43  4436.2 2266.47  4643.1 2261.18  4879.3 2256.26  4903.1 2255.55
  4978.1 2254.38  4978.3 2253.88  4981.8 2253.88  4982.1 2254.38  5022.7 2254.49
  5065.6 2255.07  5193.2 2257.72  5299.9 2259.45  5328.6 2259.67    5378 2260.68
  5392.4 2260.64    5421 2261.14  5427.5 2261.53  5435.3 2261.53  5456.1 2262.32
  5470.5 2262.37    5477 2262.76  5499.1 2263.22  5505.6 2263.61  5513.4 2263.65
  5519.9 2263.98  5527.7 2264.01  5577.2 2265.37  5704.8 2271.33  5775.7 2274.09
#Mann= 3 ,-1 , 0
  4344.7     .07       0  4978.1     .05       0  4982.1     .07       0
Bank Sta=4978.1,4982.1
XS Rating Curve= 0 ,0
Exp/Cntr=0.3,0.1

Type RM Length L Ch R = 1 ,70473   ,446,446,446
BEGIN DESCRIPTION:
Bear Creek 2 133.0
END DESCRIPTION:
XS GIS Cut Line= 3
        1800225.     13969875.04        1800225.       13969575.
      1799925.04     13969425.02
#Sta/Elev= 30
    4705 2257.11  4707.5 2257.11    4725 2256.52    4735 2255.98    4825  2250.4
    4915 2244.06    4945  2242.2    4955 2241.73    4975 2241.28  5000.5 2241.17
  5000.8 2240.67  5004.3 2240.67  5004.5 2241.17  5007.8 2241.17  5013.4 2241.39
    5019 2241.49  5049.8 2242.67  5130.8 2246.31  5183.9 2248.51    5237 2251.01
  5256.6 2251.81  5259.4 2252.01  5281.8    2253  5287.3 2253.17  5304.1 2253.97
  5309.7 2254.08  5326.5 2254.89  5332.1    2255  5337.7 2255.45  5340.4 2255.45
#Mann= 3 ,-1 , 0
    4705     .07       0  5000.5     .05       0  5004.5     .07       0
Bank Sta=5000.5,5004.5
XS Rating Curve= 0 ,0
Exp/Cntr=0.3,0.1

Type RM Length L Ch R = 1 ,70027   ,449,449,449
BEGIN DESCRIPTION:
Bear Creek 2 132.0
END DESCRIPTION:
XS GIS Cut Line= 3
        1800525.     13969624.97        1800575.       13969325.
      1800475.02     13969225.02
#Sta/Elev= 30
  4691.2 2246.29  4693.7 2246.29  4719.1 2245.28  4724.1 2245.43  4731.7 2245.14
  4779.9 2243.74  4784.9 2243.89  4840.7 2242.19  4845.8 2242.35  4901.5  2240.6
  4906.6 2240.81  4944.6 2239.21  4954.8 2238.65  4962.4  2238.1  4967.4 2236.59
    4975 2235.86  4985.2  2235.2  4990.8 2234.54    4991 2234.04  4994.5 2234.04
  4994.8 2234.54  4998.8 2234.54  5009.5 2235.59  5023.6 2235.11  5037.7 2235.32
  5051.9 2236.13  5094.3 2240.32  5108.4    2241  5133.2 2241.85  5136.7 2241.85
#Mann= 3 ,-1 , 0
  4691.2     .07       0  4990.8     .05       0  4994.8     .07       0
Bank Sta=4990.8,4994.8
XS Rating Curve= 0 ,0
Exp/Cntr=0.3,0.1

Type RM Length L Ch R = 1 ,69578   ,416,416,416
BEGIN DESCRIPTION:
Bear Creek 2 131.0
END DESCRIPTION:
XS GIS Cut Line= 3
        1800975.       13969275.        1800925.       13969125.
      1800625.04     13969025.01
#Sta/Elev= 30
  4837.9    2235  4848.4 2234.44    4859 2233.17  4869.5 2232.35  4880.1 2231.18
  4890.6 2229.37  4911.7 2228.24  4922.2 2226.98  4943.3 2225.13  4953.9 2223.84
  4993.4 2221.83  5006.6 2221.64  5015.1 2221.03  5015.3 2220.53  5018.8 2220.53
  5019.1 2221.03  5027.6 2221.86  5038.2 2222.29  5059.3 2221.26  5101.4  2223.8
    5112 2225.08    5133 2226.12  5143.6 2227.29  5175.2 2228.73  5196.3 2229.38
  5270.1 2234.18  5291.2 2234.18  5301.7 2234.56  5309.6 2235.46  5312.2 2235.46
#Mann= 3 ,-1 , 0
  4837.9     .07       0  5015.1     .05       0  5019.1     .07       0
Bank Sta=5015.1,5019.1
XS Rating Curve= 0 ,0
Exp/Cntr=0.3,0.1

Type RM Length L Ch R = 1 ,69162   ,457,457,457
BEGIN DESCRIPTION:
Bear Creek 2 130.0
END DESCRIPTION:
XS GIS Cut Line= 3
        1801225.     13968975.01        1801175.       13968875.
      1800974.98     13968574.97
#Sta/Elev= 30
  4888.2 2227.59  4963.7 2223.57  4969.3 2222.65  4972.1 2221.59  4977.7 2220.54
    4986 2217.98  4991.6 2215.77  5007.5  2216.1  5013.5 2216.71  5028.6 2217.32
  5036.1 2217.33  5064.6 2216.92  5083.6 2215.58  5083.9 2215.08  5087.4 2215.08
  5087.6 2215.58  5100.7 2216.34  5115.7 2216.48  5121.7 2217.15  5151.7 2217.78
  5157.8 2218.65  5166.8 2218.85  5172.8 2220.23  5180.3 2220.79  5202.8 2223.41
  5208.8 2224.83  5265.9 2230.04  5288.5 2231.14  5324.5 2233.54  5360.6 2234.31
#Mann= 3 ,-1 , 0
  4888.2     .07       0  5083.6     .05       0  5087.6     .07       0
Bank Sta=5083.6,5087.6
XS Rating Curve= 0 ,0
Exp/Cntr=0.3,0.1

Type RM Length L Ch R = 1 ,68705   ,445,445,445
BEGIN DESCRIPTION:
Bear Creek 2 129.0
END DESCRIPTION:
XS GIS Cut Line= 3
        1801475.     13968825.04        1801475.       13968575.
      1801375.02     13968375.04
#Sta/Elev= 30
  4749.8 2221.86  4799.8 2220.23  4809.8 2219.47  4829.8 2218.71  4899.8 2212.57
  4939.8 2211.17  4949.8 2212.42  4979.8 2211.18  4989.8 2211.07  4997.3 2210.55
  5008.2 2210.29  5013.8 2210.64  5028.6 2210.06  5028.8 2209.56  5032.3 2209.56
  5032.6 2210.06  5044.6 2210.95  5066.9 2210.99  5080.9  2210.5  5089.3 2210.64
  5097.7 2211.34  5103.3 2212.37  5111.6 2215.23    5120 2217.25  5125.6 2218.02
    5134  2219.8    5148 2221.64  5164.7 2224.19  5187.1 2226.03  5223.4 2227.73
#Mann= 3 ,-1 , 0
  4749.8     .07       0  5028.6     .05       0  5032.6     .07       0
Bank Sta=5028.6,5032.6
XS Rating Curve= 0 ,0
Exp/Cntr=0.3,0.1

Type RM Length L Ch R = 1 ,68260   ,437,437,437
BEGIN DESCRIPTION:
Bear Creek 2 128.0
END DESCRIPTION:
XS GIS Cut Line= 3
      1802125.02     13968224.99        1801825.       13968325.
        1801575.       13968275.
#Sta/Elev= 30
  4679.9 2218.43  4690.5 2218.33    4701 2217.86  4732.6 2216.02  4753.7 2213.78
  4764.2 2213.38    4817 2207.71  4827.5 2206.98  4859.1 2205.64    4954 2203.71
  4964.5  2203.3  4973.1 2202.16  4973.3 2201.66  4976.8 2201.66  4977.1 2202.16
  4985.6  2204.6  5021.6 2205.37  5036.9 2202.18  5047.1 2202.52  5077.7  2205.8
  5087.9 2206.47  5098.1  2207.5  5108.3 2207.97  5118.5 2209.43  5128.7  2210.4
  5138.9 2211.01  5159.3 2214.06  5200.1 2218.98  5220.5 2221.09  5251.1 2222.22
#Mann= 3 ,-1 , 0
  4679.9     .07       0  4973.1     .05       0  4977.1     .07       0
Bank Sta=4973.1,4977.1
XS Rating Curve= 0 ,0
Exp/Cntr=0.3,0.1

Type RM Length L Ch R = 1 ,67823   ,446,446,446
BEGIN DESCRIPTION:
Bear Creek 2 127.0
END DESCRIPTION:
XS GIS Cut Line= 3
      1802074.98       13967925.        1801925.       13967925.
      1801624.99     13968075.01
#Sta/Elev= 30
  4849.6 2210.57  4889.6 2208.02  4899.6 2206.94  4909.6 2206.63  4919.6 2205.51
  4939.6 2201.17  4949.6 2199.57  4969.6 2199.54  4989.6 2198.74    5006 2197.45
  5006.2 2196.95  5009.7 2196.95    5010 2197.45  5013.6 2197.52  5021.9 2199.27
  5030.3 2200.44  5035.9 2200.22  5044.3 2200.84  5080.6 2200.65  5147.7 2202.29
  5200.8 2202.82  5223.2 2203.59  5237.2 2204.47  5245.5 2205.42  5267.9 2209.35
  5276.3 2210.43  5312.6  2213.2  5326.6 2213.86  5332.2 2214.92    5335 2214.92
#Mann= 3 ,-1 , 0
  4849.6     .07       0    5006     .05       0    5010     .07       0
Bank Sta=5006,5010
XS Rating Curve= 0 ,0
Exp/Cntr=0.3,0.1

Type RM Length L Ch R = 1 ,67377   ,450,450,450
BEGIN DESCRIPTION:
Bear Creek 2 126.0
END DESCRIPTION:
XS GIS Cut Line= 4
      1802174.98     13967624.99        1801975.       13967525.
      1801810.02     13967546.49        1801375.       13967925.
#Sta/Elev= 30
  4768.6 2215.53  4876.6 2206.35  4911.1 2202.92  4916.7 2202.97  4933.5 2198.78
  4947.5  2197.3  4983.8 2196.18  5020.4 2195.88  5020.7 2195.38  5024.2 2195.38
  5024.4 2195.88  5029.2 2197.48  5059.9 2197.67  5133.4 2197.08    5204 2197.81
  5218.2 2198.47  5274.2 2198.59  5324.3 2199.55  5345.4  2200.9  5366.3 2201.35
  5373.9 2202.61  5380.6 2202.65  5402.4 2204.78  5423.3 2206.01  5494.5 2214.06
    5523 2216.26  5615.1 2220.43  5621.7 2221.46  5678.7 2225.33  5735.2 2227.79
#Mann= 5 ,-1 , 0
  4768.6     .07       0  4876.6      .1       0  5020.4     .05       0
  5024.4      .1       0  5059.9     .07       0
Bank Sta=5020.4,5024.4
XS Rating Curve= 0 ,0
Exp/Cntr=0.3,0.1

Type RM Length L Ch R = 1 ,66927   ,148,148,148
BEGIN DESCRIPTION:
Bear Creek 2 125.0
END DESCRIPTION:
XS GIS Cut Line= 3
      1802225.05       13967125.        1801925.       13967125.
      1801435.81     13966985.27
#Sta/Elev= 30
    4700 2210.31  4734.2 2208.26    4910 2195.22  4927.2 2192.58    4950 2191.19
    4990 2191.61  5022.1 2189.01  5041.6 2191.02    5054 2188.86  5054.2 2188.36
    5058 2188.86  5062.4 2191.76  5083.2 2190.89  5089.8 2192.55  5145.6 2193.13
  5167.8 2191.49  5201.6 2191.83  5218.4 2193.62  5301.6 2197.93  5313.4 2200.05
  5322.4  2198.7    5342 2202.19  5347.2 2201.52  5353.6 2204.31    5364 2207.01
  5386.2 2210.67  5405.6  2212.3    5420 2215.26    5459 2218.52  5508.8  2219.4
#Mann= 5 ,-1 , 0
    4700     .07       0  4734.2      .1       0  4927.2     .07       0
    5054     .05       0    5058     .07       0
Bank Sta=5054,5058
XS Rating Curve= 0 ,0
Exp/Cntr=0.3,0.1

Type RM Length L Ch R = 1 ,66779   ,201,201,201
BEGIN DESCRIPTION:
Bear Creek 2 124.2
END DESCRIPTION:
XS GIS Cut Line= 4
       1802346.8     13967101.59      1801910.65     13967010.45
      1801780.44     13966958.37      1801503.55     13966759.35
#Sta/Elev= 30
  4515.8 2212.26  4573.1 2210.45  4599.4 2207.81  4623.1 2207.35    4661 2204.84
  4698.6 2203.51  4844.6 2198.78  4946.7 2197.02  4986.6 2197.31  4999.8 2196.41
  5008.3  2190.3  5008.6  2189.8  5012.7  2190.3  5032.1 2197.82  5180.3 2202.46
  5186.4 2200.99  5201.1 2203.82  5207.3 2203.08  5215.9 2204.27    5222 2202.86
  5230.6 2205.26  5236.8 2203.26  5243.8 2206.05  5251.5 2206.73  5266.2  2207.4
  5272.4 2206.29  5287.1 2208.71  5293.2 2208.31  5301.8 2209.63  5442.6 2218.06
#Mann= 5 ,-1 , 0
  4515.8     .07       0    4661      .1       0  4698.6     .07       0
  5008.3     .05       0  5012.7     .07       0
Bank Sta=5008.3,5012.7
XS Rating Curve= 0 ,0
Exp/Cntr=0.3,0.1

Type RM Length L Ch R = 1 ,66578   ,152,152,152
BEGIN DESCRIPTION:
Bear Creek 2 124.1
END DESCRIPTION:
XS GIS Cut Line= 3
      1802431.31     13967123.17      1801949.11      13966818.9
      1801498.69     13966666.12
#Sta/Elev= 30
  4403.5 2215.23  4553.4 2212.24    4705 2207.81  4820.3 2195.32  4856.8 2193.21
  4893.3 2191.67  4899.2 2193.38  4914.4 2191.28  4920.4 2193.61  4929.7 2192.34
  4935.6 2195.41  4950.9 2191.78  4956.8 2194.65  4966.2 2192.62  4972.1 2193.91
  4988.6 2190.92  4997.6 2186.73  5007.5 2186.04  5007.8 2185.54  5011.9 2186.04
    5029 2187.16  5034.3 2190.95  5154.6 2190.83  5248.9  2195.4  5263.1 2197.27
  5280.3 2203.26  5285.5  2202.2  5311.7 2210.79  5374.5 2217.47  5449.3 2222.11
#Mann= 4 ,-1 , 0
  4403.5     .07       0  4553.4     .07       0  5007.5     .05       0
  5011.9     .07       0
Bank Sta=5007.5,5011.9
XS Rating Curve= 0 ,0
Exp/Cntr=0.3,0.1

Type RM Length L Ch R = 1 ,66426   ,391,391,391
BEGIN DESCRIPTION:
Bear Creek 2 124.0
END DESCRIPTION:
XS GIS Cut Line= 3
      1802533.59     13966962.43       1801978.4      13966691.6
      1801555.32      13966522.9
#Sta/Elev= 30
  4379.1 2216.73  4488.8 2213.48  4524.6  2210.6  4569.7 2208.28  4721.8 2201.93
  4823.1 2195.83  4862.6 2192.52  4868.1 2193.03  4878.2 2191.81  4980.8 2188.85
  4989.5 2188.28  4995.9 2186.22  5009.1 2185.32  5009.4 2184.82  5013.5 2185.32
  5043.6 2188.21  5172.7 2188.83  5188.9 2190.25  5219.2 2190.69  5258.9 2193.46
  5297.3 2199.26  5302.7 2199.26    5327 2203.89  5334.2 2206.24  5351.3 2209.08
  5356.6 2209.06  5375.5 2212.15  5380.9 2211.88  5405.2 2216.27  5452.3 2219.25
#Mann= 3 ,-1 , 0
  4379.1     .07       0  5009.1     .05       0  5013.5     .07       0
Bank Sta=5009.1,5013.5
XS Rating Curve= 0 ,0
Exp/Cntr=0.3,0.1

Type RM Length L Ch R = 1 ,66035   ,464,464,464
BEGIN DESCRIPTION:
Bear Creek 2 123.0
END DESCRIPTION:
XS GIS Cut Line= 3
      1802450.23     13966501.61        1801975.       13966325.
        1801575.       13966425.
#Sta/Elev= 30
  4498.9 2201.82  4587.1 2197.51  4622.8 2195.11  4717.8 2190.86  4813.9 2189.13
  4844.3 2187.78  4874.6 2185.31  4920.5 2186.11  4963.4 2184.02  4963.8 2183.52
  4967.6 2183.52  4967.9 2184.02    4996    2185  5016.2 2184.14  5023.9 2184.76
  5029.1 2184.19  5036.8 2185.99  5047.1 2186.62  5139.9 2189.19  5235.2  2195.4
  5271.3 2199.29  5276.5 2199.32  5284.2 2200.98  5312.5 2205.01  5317.7 2205.12
  5325.4 2206.86  5353.8 2210.53  5358.9 2210.58    5395 2215.31  5418.2 2217.03
#Mann= 3 ,-1 , 0
  4498.9     .07       0  4963.4     .05       0  4967.9     .07       0
Bank Sta=4963.4,4967.9
XS Rating Curve= 0 ,0
Exp/Cntr=0.3,0.1

Type RM Length L Ch R = 1 ,65571   ,469,469,469
BEGIN DESCRIPTION:
Bear Creek 2 122.0
END DESCRIPTION:
XS GIS Cut Line= 3
      1802424.99     13966024.99        1802175.       13965925.
        1801375.       13966175.
#Sta/Elev= 30
  4725.5 2195.65  4794.1 2193.38    4848 2190.65  4896.5 2187.16  4901.8 2187.31
  4950.3 2183.27  4955.7 2183.52  4970.9 2178.49  4971.3 2177.99  4975.2 2177.99
  4975.5 2178.49  4979.9 2180.18  5005.2 2179.98    5011 2179.19  5016.2  2180.1
  5026.2 2179.08  5043.5  2181.6  5204.3 2184.36  5281.3 2186.11  5313.8 2187.43
  5346.2 2189.83  5448.9 2195.13  5476.2 2197.29  5481.4  2196.7  5539.5 2201.44
  5560.5 2204.25  5623.4 2210.03  5759.6 2219.81  5801.5 2222.52  5832.9 2223.68
#Mann= 3 ,-1 , 0
  4725.5     .07       0  4970.9     .05       0  4975.5     .07       0
Bank Sta=4970.9,4975.5
XS Rating Curve= 0 ,0
Exp/Cntr=0.3,0.1

Type RM Length L Ch R = 1 ,65102   ,449,449,449
BEGIN DESCRIPTION:
Bear Creek 2 121.0
END DESCRIPTION:
XS GIS Cut Line= 3
      1802424.95     13965524.99        1802125.       13965475.
        1801725.       13965825.
#Sta/Elev= 30
    4696 2190.39  4756.8 2188.55  4789.7 2187.99  4888.6 2184.15  4906.3 2182.77
  4911.4 2182.73  4929.1 2180.24  4959.5 2174.92  4972.2 2174.26  5003.4 2174.62
  5025.7 2173.82  5026.1 2173.32  5030.1 2173.32  5030.4 2173.82  5035.7 2176.14
  5042.3 2176.39  5049.9 2178.35  5127.7 2180.27  5162.9 2180.34  5184.7 2181.15
  5205.6 2181.41  5212.7 2180.69  5219.8 2180.72  5226.5 2180.95    5234 2181.97
  5276.8 2183.83  5311.9 2184.49  5340.4 2185.87  5418.2 2188.51  5531.6 2193.73
#Mann= 3 ,-1 , 0
    4696     .07       0  5025.7     .05       0  5030.4     .07       0
Bank Sta=5025.7,5030.4
XS Rating Curve= 0 ,0
Exp/Cntr=0.3,0.1

Type RM Length L Ch R = 1 ,64653   ,478,478,478
BEGIN DESCRIPTION:
Bear Creek 2 120.0
END DESCRIPTION:
XS GIS Cut Line= 3
      1802475.01       13965125.        1802075.       13965075.
      1801675.02     13965324.99
#Sta/Elev= 30
  4596.4 2187.84  4727.4 2182.36  4918.9 2176.76  4939.1 2175.43  4949.1 2174.33
  4956.7 2172.83  4961.7 2172.94  4969.3 2172.29  4979.4 2171.99    4987 2170.99
  4987.4 2170.49  4991.5 2170.49  4991.8 2170.99    4997 2171.79  5002.5 2171.79
  5007.2 2172.43  5028.4 2173.17  5034.9 2174.56  5058.5 2175.68  5129.2    2176
  5201.8 2177.23  5223.6 2176.94  5253.7 2177.99  5282.5 2178.35  5290.2 2178.86
  5296.1 2178.66  5332.7 2180.42  5384.5 2183.92  5442.3 2186.38  5471.2 2187.15
#Mann= 3 ,-1 , 0
  4596.4     .07       0    4987     .05       0  4991.8     .07       0
Bank Sta=4987,4991.8
XS Rating Curve= 0 ,0
Exp/Cntr=0.3,0.1

Type RM Length L Ch R = 1 ,64175   ,482,482,482
BEGIN DESCRIPTION:
Bear Creek 2 119.0
END DESCRIPTION:
XS GIS Cut Line= 3
      1802475.01     13964875.01        1802075.       13964625.
      1801624.96     13964825.02
#Sta/Elev= 30
  4528.7 2186.27  4557.6 2184.92  4564.1 2184.16  4578.8 2183.66  4594.2 2182.13
  4615.4 2181.21  4630.7 2179.93  4725.1 2175.96  4898.4  2172.4  4956.2 2171.74
  4977.4 2170.57  4986.8 2169.52  4992.7 2169.66    4995 2169.02  4995.4 2168.52
  4999.6 2168.52  4999.9 2169.02  5014.8 2169.07  5032.6 2169.83  5055.1 2169.65
  5061.3 2170.93  5084.5 2171.57  5142.7 2171.98  5165.2 2173.32    5183 2175.07
  5258.3 2178.53  5317.8 2180.41  5408.7 2182.12  5478.5 2184.56  5492.9 2184.64
#Mann= 3 ,-1 , 0
  4528.7     .07       0    4995     .05       0  4999.9     .07       0
Bank Sta=4995,4999.9
XS Rating Curve= 0 ,0
Exp/Cntr=0.3,0.1

Type RM Length L Ch R = 1 ,63693   ,471,471,471
BEGIN DESCRIPTION:
Bear Creek 2 118.0
END DESCRIPTION:
XS GIS Cut Line= 3
      1802475.05       13964175.        1802175.       13964175.
      1801574.99     13963624.99
#Sta/Elev= 30
    4705 2183.24    4855 2174.25    4865  2172.9    4935 2166.93    4945 2166.55
    4955 2167.25    4965  2166.8    4975 2165.15    4985  2165.7    5000 2165.06
  5000.4 2164.56  5004.6 2164.56    5005 2165.06  5054.7 2166.65  5061.5 2166.37
  5068.9 2167.21  5097.2 2168.28  5174.9 2169.09  5181.7 2168.77  5189.1 2169.38
  5252.6 2167.91  5302.6 2168.55  5316.7 2167.79  5323.5 2166.78  5401.2 2168.77
  5429.6 2169.91  5472.1 2172.98  5578.2  2181.6  5726.8 2188.26    5819 2190.72
#Mann= 3 ,-1 , 0
    4705     .07       0    5000     .05       0    5005     .07       0
Bank Sta=5000,5005
XS Rating Curve= 0 ,0
Exp/Cntr=0.3,0.1

Type RM Length L Ch R = 1 ,63222   ,438,438,438
BEGIN DESCRIPTION:
Bear Creek 2 117.0
END DESCRIPTION:
XS GIS Cut Line= 3
      1802475.01     13963975.01        1802175.       13963725.
      1801775.03     13963575.01
#Sta/Elev= 30
    4622 2180.77  4678.6 2177.85  4735.9 2173.61  4799.7 2171.98    4814 2172.34
  4863.5 2169.06  4927.3 2166.02  4941.6 2163.55  4948.1 2163.38  4955.9 2161.71
  4970.2 2161.18  4991.1 2161.89  5002.6 2161.14  5003.1 2160.64  5007.7 2160.64
  5008.1 2161.14  5044.6 2163.86  5107.8 2165.51  5173.6 2166.19  5215.5 2167.74
  5228.8 2169.71  5247.5 2170.76  5253.7 2172.19  5259.1 2172.39  5290.2 2176.61
  5314.2 2178.19  5339.2 2181.04  5369.4  2182.7  5394.3 2184.81  5439.7 2186.86
#Mann= 3 ,-1 , 0
    4622     .07       0  5002.6     .05       0  5008.1     .07       0
Bank Sta=5002.6,5008.1
XS Rating Curve= 0 ,0
Exp/Cntr=0.3,0.1

Type RM Length L Ch R = 1 ,62784   ,450,450,450
BEGIN DESCRIPTION:
Bear Creek 2 116.0
END DESCRIPTION:
XS GIS Cut Line= 3
      1802575.03     13963725.03        1802175.       13963325.
      1801974.98     13963375.01
#Sta/Elev= 30
  4433.9 2175.33  4532.9 2172.06  4589.5 2170.75  4646.1 2168.52  4752.1 2166.08
  4801.6 2163.53  4900.6 2160.28  4957.2 2161.37  4971.3 2161.18  4985.5 2160.59
  4996.1 2159.61  5002.2 2159.61  5007.2 2158.21  5007.6 2157.71  5012.2 2157.71
  5012.7 2158.21  5017.7 2159.17  5022.8  2159.5  5030.5 2160.77  5040.9 2161.87
  5082.1 2165.32  5092.4 2165.86  5100.1 2167.14  5105.3 2167.01  5141.4 2171.52
  5146.5  2171.6  5182.6 2176.25  5187.7 2176.18  5195.5 2177.02  5205.8 2177.37
#Mann= 3 ,-1 , 0
  4433.9     .07       0  5007.2     .05       0  5012.7     .07       0
Bank Sta=5007.2,5012.7
XS Rating Curve= 0 ,0
Exp/Cntr=0.3,0.1

Type RM Length L Ch R = 1 ,62334   ,451,451,451
BEGIN DESCRIPTION:
Bear Creek 2 115.0
END DESCRIPTION:
XS GIS Cut Line= 3
      1802724.97     13963324.97        1802325.       13962925.
      1801925.05       13962925.
#Sta/Elev= 30
  4439.4  2171.6  4474.7 2170.73  4693.9 2163.22  4764.6 2161.32  4849.5  2159.8
  4863.6 2160.03  4920.2 2159.13  4962.6    2156  4990.9 2155.77  5012.2 2154.75
  5012.7 2154.25  5017.4 2154.25  5017.8 2154.75    5025 2156.76    5045 2159.41
    5065 2160.22    5075 2161.01    5105 2164.19    5185 2167.52    5195  2168.4
    5205 2168.31    5255 2170.33    5295 2172.71    5305 2172.86    5325 2172.06
    5345 2175.64    5365 2177.85    5375 2178.79    5385 2179.07    5405 2180.52
#Mann= 3 ,-1 , 0
  4439.4     .07       0  5012.2     .05       0  5017.8     .07       0
Bank Sta=5012.2,5017.8
XS Rating Curve= 0 ,0
Exp/Cntr=0.3,0.1

Type RM Length L Ch R = 1 ,61883   ,482,482,482
BEGIN DESCRIPTION:
Bear Creek 2 114.0
END DESCRIPTION:
XS GIS Cut Line= 3
      1803275.01       13962625.        1802475.       13962525.
      1802075.04     13962624.99
#Sta/Elev= 30
  4194.1 2179.32  4264.7 2176.19  4274.7 2176.26  4312.5  2172.5  4335.2 2171.43
  4398.2 2170.02  4456.1 2167.15  4486.4 2166.97  4499.9 2166.22  4590.8 2163.48
  4657.7 2160.93  4768.5 2158.82  4869.3 2154.56  4939.9 2156.62  4962.5 2155.74
  4980.2 2153.49    4995 2153.37  4995.5 2152.87  5000.2 2152.87  5000.6 2153.37
  5041.6 2154.22  5134.3 2159.37  5175.6 2161.06  5216.8 2161.81  5247.7 2164.04
    5289 2165.85  5348.2  2167.3  5353.4 2166.93  5361.1 2167.85  5412.6 2169.65
#Mann= 5 ,-1 , 0
  4194.1     .07       0  4499.9      .1       0  4590.8     .07       0
    4995     .05       0  5000.6     .07       0
Bank Sta=4995,5000.6
XS Rating Curve= 0 ,0
Exp/Cntr=0.3,0.1

Type RM Length L Ch R = 1 ,61401   ,447,447,447
BEGIN DESCRIPTION:
Bear Creek 2 113.0
END DESCRIPTION:
XS GIS Cut Line= 3
      1802974.97     13962374.97        1802575.       13962075.
      1801774.99     13962475.01
#Sta/Elev= 30
    4500 2165.01    4600 2160.49  4815.9 2154.61  4858.2 2153.13  4907.2  2149.9
  4928.1 2150.14  4936.4 2151.72  4963.5 2152.81  4978.1 2152.14  4993.9 2148.89
  4994.4 2148.39  4999.7 2148.89  5013.9 2149.06  5030.7 2150.78  5036.3 2150.25
  5044.7 2151.71  5075.4 2153.08  5148.1 2154.58  5187.2 2155.94  5192.8  2156.9
  5223.6 2156.43  5245.9 2157.55  5424.8 2159.48  5505.9 2163.75    5545 2164.13
  5662.4 2168.14  5701.5 2168.38    5791 2175.75  5863.6 2179.61  5894.4 2180.03
#Mann= 5 ,-1 , 0
    4500     .07       0  4815.9      .1       0  4858.2     .07       0
  4993.9     .05       0  4999.7     .07       0
Bank Sta=4993.9,4999.7
XS Rating Curve= 0 ,0
Exp/Cntr=0.3,0.1

Type RM Length L Ch R = 1 ,60954   ,466,466,466
BEGIN DESCRIPTION:
Bear Creek 2 112.0
END DESCRIPTION:
XS GIS Cut Line= 3
      1803174.98     13961974.99        1802825.       13961725.
      1802024.98     13961074.98
#Sta/Elev= 30
  4565.5 2163.41  4614.6 2162.57    4665 2159.33  4730.2  2158.3    4810 2155.59
  4946.4 2152.38  4982.1 2150.09  5002.8 2147.55    5038 2148.11  5081.1 2150.57
  5156.7  2150.7  5266.2 2148.39  5322.4 2144.23  5348.2  2143.4  5348.7  2142.9
  5354.1  2143.4  5365.5 2145.69    5372 2145.58  5379.9 2147.45  5407.9 2148.64
  5472.3 2148.22  5571.7 2149.59  5670.8 2152.67  5713.9 2156.07  5749.1 2157.81
  5798.7 2158.54  5856.1 2160.63  5891.3 2160.77  5934.4 2162.71  6026.4 2164.78
#Mann= 3 ,-1 , 0
  4565.5     .07       0  5348.2     .05       0  5354.1     .07       0
Bank Sta=5348.2,5354.1
XS Rating Curve= 0 ,0
Exp/Cntr=0.3,0.1

Type RM Length L Ch R = 1 ,60488   ,463,463,463
BEGIN DESCRIPTION:
Bear Creek 2 111.0
END DESCRIPTION:
XS GIS Cut Line= 3
        1803225.       13961675.        1802875.       13961275.
      1802074.97     13961024.99
#Sta/Elev= 30
  4462.8 2159.67  4547.8 2159.05  4696.8 2154.59  4809.7 2153.32  4880.9 2149.72
  4937.8 2148.53  4952.1 2147.44  4958.7 2145.98    4973 2144.95  4987.2 2145.26
    4991 2144.18  5004.8 2144.93  5010.6 2146.11  5048.3 2145.99  5075.5 2147.42
  5161.9  2147.5  5253.2  2142.8  5253.7  2142.3  5259.2  2142.8  5308.1 2145.12
  5351.1 2146.04  5434.3 2150.58    5481 2151.22  5513.4 2154.03  5551.2 2155.53
  5616.1 2156.52  5696.3 2159.86  5751.3 2160.92  5790.6 2163.05  5832.5 2163.73
#Mann= 3 ,-1 , 0
  4462.8     .07       0  5253.2     .05       0  5259.2     .07       0
Bank Sta=5253.2,5259.2
XS Rating Curve= 0 ,0
Exp/Cntr=0.3,0.1

Type RM Length L Ch R = 1 ,60025   ,422,422,422
BEGIN DESCRIPTION:
Bear Creek 2 110.0
END DESCRIPTION:
XS GIS Cut Line= 3
        1803375.       13961175.        1802975.       13960875.
      1802175.01     13960175.01
#Sta/Elev= 30
  4495.1 2155.67    4667 2149.93    4767 2148.09  4845.1 2143.81  4908.6 2142.57
  4958.6 2142.77    4992 2139.93  5002.2 2139.89  5023.1 2142.33  5051.6 2143.68
    5137 2143.14  5186.3 2140.92  5232.7 2136.99  5233.2 2136.49  5238.7 2136.99
  5257.5 2138.44  5264.2 2140.28  5278.4 2141.73  5327.8 2145.56  5370.5  2145.9
  5427.4 2149.98  5484.4 2152.54    5640 2156.01  5682.7 2160.15  5725.4 2162.18
  5795.7 2163.29  5852.6 2165.84  5951.8 2168.14  6001.6 2172.72  6058.1  2176.5
#Mann= 3 ,-1 , 0
  4495.1     .07       0  5232.7     .05       0  5238.7     .07       0
Bank Sta=5232.7,5238.7
XS Rating Curve= 0 ,0
Exp/Cntr=0.3,0.1

Type RM Length L Ch R = 1 ,59603   ,449,449,449
BEGIN DESCRIPTION:
Bear Creek 2 109.0
END DESCRIPTION:
XS GIS Cut Line= 3
      1803525.03     13960725.02        1803175.       13960525.
      1802475.05     13960275.02
#Sta/Elev= 30
  4592.8  2152.5    4731 2148.98  4805.2 2145.22    4821 2143.45  4848.4 2141.86
  4915.3 2140.09  4944.8 2137.87  4998.6  2137.4  5011.3 2136.06  5042.1 2138.25
  5059.7 2140.27  5080.9 2140.53  5091.5 2140.09  5103.7 2137.48  5131.5 2133.78
    5132 2133.28  5137.1 2133.28  5137.6 2133.78  5176.5 2134.71  5221.6  2138.8
  5261.4  2140.6  5277.9 2142.46  5303.4 2143.97  5370.3 2144.75  5431.8 2148.78
  5518.9 2151.82  5537.5 2153.07  5611.8 2154.82  5675.5 2159.29  5739.2 2161.62
#Mann= 3 ,-1 , 0
  4592.8     .07       0  5131.5     .05       0  5137.6     .07       0
Bank Sta=5131.5,5137.6
XS Rating Curve= 0 ,0
Exp/Cntr=0.3,0.1

Type RM Length L Ch R = 1 ,59154   ,466,466,466
BEGIN DESCRIPTION:
Bear Creek 2 108.0
END DESCRIPTION:
XS GIS Cut Line= 4
      1803500.12     13960400.12        1803425.       13960325.
        1803225.       13960125.      1802974.98       13960125.
#Sta/Elev= 30
    4616 2146.45  4736.4 2142.87  4750.5 2141.34  4764.7 2140.92    4793  2139.1
  4807.1 2138.46  4835.4 2137.86  4849.5 2136.57  4877.8  2135.7  4920.2 2132.79
  4934.4 2131.31  4972.2 2126.39  4972.7 2125.89    4981 2125.89  4981.5 2126.39
  4990.9 2127.97  5007.6 2128.33  5025.1 2130.58  5035.1 2130.42  5045.1 2132.07
  5055.1 2133.01  5065.1 2133.52  5075.1 2134.71  5095.1 2135.25  5115.1 2136.44
  5165.1 2137.81  5205.1  2140.3  5225.1 2141.05  5245.1 2141.39  5255.1 2142.01
#Mann= 3 ,-1 , 0
    4616     .07       0  4972.2     .05       0  4981.5     .07       0
Bank Sta=4972.2,4981.5
XS Rating Curve= 0 ,0
Exp/Cntr=0.3,0.1

Type RM Length L Ch R = 1 ,58688   ,439,439,439
BEGIN DESCRIPTION:
Bear Creek 2 107.0
END DESCRIPTION:
XS GIS Cut Line= 4
      1803891.93      13960150.2        1803525.       13959875.
        1803325.       13959725.      1803224.97       13959725.
#Sta/Elev= 30
  4291.3 2145.03    4300 2145.18  4313.5 2144.13  4328.1 2143.82    4400  2142.8
  4421.8 2143.07  4428.1 2142.08  4463.5 2140.98  4571.8 2138.68  4671.8 2138.08
  4728.1 2136.54  4771.8 2136.28  4907.3 2128.95  4913.5 2128.96  4921.8 2128.32
  4942.7 2124.27    4950 2124.76  4963.5 2123.95  4971.8 2124.68  4992.7 2122.61
  4996.8 2121.34  5005.2 2120.87  5005.7 2120.37  5014.2 2120.37  5014.7 2120.87
    5020 2121.07    5030 2125.96    5040 2135.12    5050 2136.54    5100  2140.3
#Mann= 3 ,-1 , 0
  4291.3     .07       0  5005.2     .05       0  5014.7     .07       0
Bank Sta=5005.2,5014.7
XS Rating Curve= 0 ,0
Exp/Cntr=0.3,0.1

Type RM Length L Ch R = 1 ,58249   ,421,421,421
BEGIN DESCRIPTION:
Bear Creek 2 106.0
END DESCRIPTION:
XS GIS Cut Line= 3
      1803921.38     13960060.11        1803625.       13959425.
      1803574.98     13959324.97
#Sta/Elev= 30
  4299.1 2142.77  4443.5  2138.2    4449 2138.88  4525.4 2137.18  4557.8 2136.99
  4569.6 2137.47  4631.9 2135.74  4637.4 2136.16  4735.1 2135.11  4757.2 2134.36
  4774.5 2134.45    4780 2135.14  4797.4 2133.79  4802.9 2133.91  4820.2 2132.55
  4825.8 2132.69  4871.5 2130.13  4922.7 2125.43  4955.8  2123.4  4968.4 2119.73
  4991.3 2119.71  5003.5 2118.35    5004 2117.85  5012.6 2117.85  5013.1 2118.35
  5022.3 2119.56  5053.1  2129.7  5075.4 2134.31    5081 2136.26  5111.8 2137.85
#Mann= 3 ,-1 , 0
  4299.1     .07       0  5003.5     .05       0  5013.1     .07       0
Bank Sta=5003.5,5013.1
XS Rating Curve= 0 ,0
Exp/Cntr=0.3,0.1

Type RM Length L Ch R = 1 ,57828   ,604,604,604
BEGIN DESCRIPTION:
Bear Creek 2 105.0
END DESCRIPTION:
XS GIS Cut Line= 4
      1803962.99     13960062.09      1804002.02      13959564.6
        1803975.       13959225.        1803925.     13959124.99
#Sta/Elev= 30
  4164.8 2143.56    4202 2141.75  4312.3 2140.09  4352.5 2138.09  4384.9  2138.1
  4392.6 2137.53  4502.9 2135.71    4543 2133.22  4613.3 2131.78  4623.3 2132.01
  4633.1 2131.32  4661.1 2130.82  4713.6 2130.51  4733.6 2129.26  4817.2  2126.5
    4854 2124.02  4884.1 2123.84  4945.4 2120.52  4979.6 2116.57  4980.1 2116.07
  4988.7 2116.07  4989.2 2116.57  4994.5 2117.01    5002 2118.51  5007.3 2118.51
  5012.9 2121.52  5018.5 2122.51  5035.2 2128.17    5080  2132.9  5116.3 2134.35
#Mann= 3 ,-1 , 0
  4164.8     .07       0  4979.6     .05       0  4989.2     .07       0
Bank Sta=4979.6,4989.2
XS Rating Curve= 0 ,0
Exp/Cntr=0.3,0.1

Type RM Length L Ch R = 1 ,57224   ,305,305,305
BEGIN DESCRIPTION:
Bear Creek 2 104.0
END DESCRIPTION:
XS GIS Cut Line= 3
        1804675.       13959425.      1804498.61     13959113.32
      1804074.98     13958874.99
#Sta/Elev= 30
  4704.6 2138.56  4734.2 2137.41  4755.8 2134.69  4771.7 2133.96    4785 2132.64
    4815 2131.57  4858.3  2126.9  4888.4 2125.55  4895.8 2125.76  4901.6 2124.58
  4960.8 2118.88  4971.6 2117.13  4972.1 2116.63  4981.2 2116.63  4981.7 2117.13
  4991.9 2117.25  4998.3 2118.24  5014.2 2118.58  5167.9 2118.65  5189.6 2120.78
  5195.3 2121.96  5211.3 2122.92    5217 2124.27    5233  2126.3  5276.3 2128.61
  5319.6  2130.2  5373.2 2130.52  5519.1 2134.22  5535.1 2135.19  5548.8 2135.05
#Mann= 3 ,-1 , 0
  4704.6     .07       0  4971.6     .05       0  4981.7     .07       0
Bank Sta=4971.6,4981.7
XS Rating Curve= 0 ,0
Exp/Cntr=0.3,0.1

Type RM Length L Ch R = 1 ,56919   ,441,441,441
BEGIN DESCRIPTION:
Bear Creek 2 103.0
END DESCRIPTION:
XS GIS Cut Line= 3
      1804875.02     13959125.01        1804775.       13959075.
      1804425.03     13958825.02
#Sta/Elev= 30
  4894.6 2134.91  4925.4 2132.87  4939.3 2128.66  4947.7 2124.93  4953.3 2120.14
  4961.7 2116.21  4970.1 2113.79  4984.1 2112.49  4992.4 2112.53  4992.9 2112.08
  4993.4 2111.58  5002.6 2111.58  5003.1 2112.08  5003.6 2112.72  5013.8 2113.14
  5019.9 2115.63  5043.3 2117.51  5064.2 2117.28  5078.9 2117.63  5085.1 2118.34
    5106 2118.15  5129.3 2118.98  5257.1 2120.89  5271.9  2122.2  5286.6 2122.18
    5337 2124.15    5364 2126.18  5387.4 2127.11  5414.4 2129.17  5436.5  2130.2
#Mann= 3 ,-1 , 0
  4894.6     .07       0  4992.9     .05       0  5003.1     .07       0
Bank Sta=4992.9,5003.1
XS Rating Curve= 0 ,0
Exp/Cntr=0.3,0.1

Type RM Length L Ch R = 1 ,56478   ,471,471,471
BEGIN DESCRIPTION:
Bear Creek 2 102.0
END DESCRIPTION:
XS GIS Cut Line= 3
      1805175.03     13958825.01        1805075.       13958775.
      1804875.02     13958375.04
#Sta/Elev= 30
  4888.4 2135.05  4896.8 2134.45  4919.2 2130.75  4941.5 2128.46  4955.5 2125.92
  4969.5  2121.6  4977.9 2118.27  4986.3 2112.73  4991.9 2110.17    4992 2109.33
  4992.5 2108.83  5002.3 2108.83  5002.8 2109.33  5014.2 2109.68  5022.6 2111.07
    5045 2110.98  5053.3 2110.26  5058.9  2111.2  5081.3 2111.78  5089.7 2111.39
  5134.4 2113.79  5223.8 2115.19  5276.9 2118.35  5304.9 2118.99  5366.4 2124.49
    5372 2124.39  5388.8 2125.69  5394.3 2126.68  5439.1 2129.01  5447.4 2128.97
#Mann= 3 ,-1 , 0
  4888.4     .07       0    4992     .05       0  5002.8     .07       0
Bank Sta=4992,5002.8
XS Rating Curve= 0 ,0
Exp/Cntr=0.3,0.1

Type RM Length L Ch R = 1 ,56007   ,462,462,462
BEGIN DESCRIPTION:
Bear Creek 2 101.0
END DESCRIPTION:
XS GIS Cut Line= 3
      1805474.97     13958474.98        1805275.       13958375.
      1804925.02       13958325.
#Sta/Elev= 30
  4776.1 2129.11  4784.4 2129.25  4812.4 2126.81  4820.8 2124.65  4829.2 2123.15
  4851.5  2120.6  4865.5 2119.46  4901.8 2112.43  4910.2 2111.46  4924.2  2110.7
    4941 2109.01  4963.3 2109.33  4980.2 2108.86  4980.7 2108.36  4990.6 2108.36
  4991.1 2108.86  4996.9 2109.72  5009.8 2109.89  5019.9 2109.49  5040.1 2110.24
  5050.2 2110.09  5070.4 2111.06  5100.7 2110.78  5110.8 2111.56  5120.9 2111.83
  5272.4 2124.34  5312.8 2127.29  5322.9 2128.36  5343.1 2129.76  5353.2 2129.86
#Mann= 3 ,-1 , 0
  4776.1     .07       0  4980.2     .05       0  4991.1     .07       0
Bank Sta=4980.2,4991.1
XS Rating Curve= 0 ,0
Exp/Cntr=0.3,0.1

Type RM Length L Ch R = 1 ,55545   ,468,468,468
BEGIN DESCRIPTION:
Bear Creek 2 100.0
END DESCRIPTION:
XS GIS Cut Line= 3
      1805775.03     13958125.01        1805425.       13957975.
      1805325.03     13957875.03
#Sta/Elev= 30
  4623.7 2128.32  4656.4 2127.57  4685.4 2123.21  4690.8 2123.12  4714.4 2120.04
  4761.5 2111.87  4790.6 2109.08  4819.6 2108.13  4837.7 2108.71    4874 2108.15
  4884.9 2108.89  4895.7 2108.25  4913.9 2108.66  4937.4 2107.35  4950.1 2107.29
    4961 2106.48  4971.9 2103.96    4990 2100.57  4996.4  2099.9  4996.9  2099.4
  5006.8  2099.4  5007.3  2099.9  5008.1  2099.9  5018.7 2104.73  5032.8 2110.24
  5039.9 2110.53    5047 2111.66  5117.7 2116.18  5131.8 2117.65  5145.9 2118.08
#Mann= 3 ,-1 , 0
  4623.7     .07       0  4996.4     .05       0  5007.3     .07       0
Bank Sta=4996.4,5007.3
XS Rating Curve= 0 ,0
Exp/Cntr=0.3,0.1

Type RM Length L Ch R = 1 ,55077   ,478,478,478
BEGIN DESCRIPTION:
Bear Creek 2 99.0
END DESCRIPTION:
XS GIS Cut Line= 3
      1805925.01     13958025.03        1805725.       13957625.
      1805524.99     13957424.99
#Sta/Elev= 30
  4552.4 2130.04  4597.2 2127.82  4619.5 2125.59  4655.8  2122.7    4695 2119.87
  4722.9  2118.7  4739.7 2117.48  4745.3 2116.44  4762.1 2114.95  4767.7 2113.94
  4812.4 2108.46  4896.2 2104.71  4918.6 2100.36  4924.2 2099.94  4932.6 2099.78
  4985.7 2101.75  4991.3 2099.34  4991.8 2098.84  5001.8 2098.84  5002.3 2099.34
  5013.8 2099.52  5042.1  2106.8  5056.2 2108.56  5098.6 2111.43  5141.1 2114.97
  5169.3 2118.39  5183.5 2119.55  5254.2    2129    5279 2131.44  5282.5 2131.44
#Mann= 3 ,-1 , 0
  4552.4     .07       0  4991.3     .05       0  5002.3     .07       0
Bank Sta=4991.3,5002.3
XS Rating Curve= 0 ,0
Exp/Cntr=0.3,0.1

Type RM Length L Ch R = 1 ,54599   ,453,453,453
BEGIN DESCRIPTION:
Bear Creek 2 98.0
END DESCRIPTION:
XS GIS Cut Line= 3
        1806225.       13957725.        1806075.       13957375.
      1805825.03     13957225.02
#Sta/Elev= 30
  4619.2 2116.12  4628.3 2116.21  4633.7 2115.49  4680.9 2112.63  4738.9 2110.62
  4833.2 2108.79  4838.6 2109.01  4891.2 2107.36  4956.5 2106.28  4978.2 2102.19
  4990.9 2099.05  4997.3  2098.2  5017.8 2098.09  5018.3 2097.59  5028.4 2097.59
  5028.9 2098.09  5066.1 2101.09  5093.3 2101.51  5116.6  2101.3  5124.4 2101.68
  5139.9 2103.37  5151.6 2106.34  5161.3 2107.36  5174.9 2110.56  5198.2 2114.63
  5209.9 2117.56  5233.2 2122.13  5256.6 2124.21  5268.2 2126.79  5291.5 2128.16
#Mann= 3 ,-1 , 0
  4619.2     .07       0  5017.8     .05       0  5028.9     .07       0
Bank Sta=5017.8,5028.9
XS Rating Curve= 0 ,0
Exp/Cntr=0.3,0.1

Type RM Length L Ch R = 1 ,54146   ,476,476,476
BEGIN DESCRIPTION:
Bear Creek 2 97.0
END DESCRIPTION:
XS GIS Cut Line= 3
        1806375.     13957874.97        1806325.       13957075.
      1806275.02     13956975.03
#Sta/Elev= 30
  4198.1 2120.94  4228.1 2119.09  4288.3 2117.55  4378.4 2113.46  4398.5 2113.62
  4468.6 2110.71  4518.7 2109.77  4578.8 2109.59    4649 2107.48    4669 2107.71
    4689 2106.13  4779.2 2105.06  4819.3 2103.74  4849.3 2101.98  4889.4 2097.63
  4899.4 2097.52    4917 2098.48  4949.5  2098.5  4991.6 2096.44  4992.1 2095.94
  5002.2 2095.94  5002.7 2096.44    5022 2098.13  5030.4 2101.06    5036  2102.3
  5044.4 2106.81  5058.3 2110.86  5075.1 2112.47  5097.5 2116.19  5111.4 2117.51
#Mann= 3 ,-1 , 0
  4198.1     .07       0  4991.6     .05       0  5002.7     .07       0
Bank Sta=4991.6,5002.7
XS Rating Curve= 0 ,0
Exp/Cntr=0.3,0.1

Type RM Length L Ch R = 1 ,53670   ,487,487,487
BEGIN DESCRIPTION:
Bear Creek 2 96.0
END DESCRIPTION:
XS GIS Cut Line= 3
      1806504.99     13957830.61        1806725.       13956875.
      1806675.01     13956775.01
#Sta/Elev= 30
  4018.9 2117.78  4131.4 2115.39  4174.2  2113.2  4188.8  2113.5  4250.4 2111.18
  4383.8 2109.41  4446.4 2106.02  4476.2 2105.81    4548 2102.73  4622.8 2101.13
    4784 2100.37  4799.2 2100.52  4804.5 2101.68  4825.1 2098.78  4907.2 2096.83
  4927.6 2094.85  4932.7 2095.98  4937.9 2094.84  4980.7 2092.63  4983.6 2090.64
  4984.1 2090.14  4994.8 2090.64  4996.9 2091.78  5002.3 2091.78  5007.9 2097.96
  5013.5 2099.72  5021.9 2104.42  5030.3 2106.97  5052.6 2110.06  5111.3 2114.61
#Mann= 3 ,-1 , 0
  4018.9     .07       0  4983.6     .05       0  4994.8     .07       0
Bank Sta=4983.6,4994.8
XS Rating Curve= 0 ,0
Exp/Cntr=0.3,0.1

Type RM Length L Ch R = 1 ,53183   ,470,470,470
BEGIN DESCRIPTION:
Bear Creek 2 95.0
END DESCRIPTION:
XS GIS Cut Line= 3
      1807744.88     13957004.78        1807175.       13956775.
      1806725.03     13956375.03
#Sta/Elev= 30
  4385.5 2117.29  4579.5 2114.16  4590.5 2112.95  4609.3 2112.93  4644.2 2110.14
  4716.7 2107.45  4730.4 2107.76  4794.6 2103.62  4838.2 2097.19  4892.1 2094.56
  4907.3 2092.57  4931.5 2092.18  4967.6 2087.92  4982.9 2087.04  4983.4 2086.54
  4998.2 2087.04    5000 2088.42  5013.8 2089.78    5028 2092.56  5078.1 2095.86
  5176.8  2098.4    5283 2102.47  5347.4  2109.8    5375 2111.28    5411 2116.12
  5474.5 2120.51  5488.7 2123.15  5545.6 2128.09    5574 2131.51    5602 2132.57
#Mann= 3 ,-1 , 0
  4385.5     .07       0  4982.9     .05       0  4998.2     .07       0
Bank Sta=4982.9,4998.2
XS Rating Curve= 0 ,0
Exp/Cntr=0.3,0.1

Type RM Length L Ch R = 1 ,52713   ,469,469,469
BEGIN DESCRIPTION:
Bear Creek 2 94.0
END DESCRIPTION:
XS GIS Cut Line= 3
      1807675.02     13956775.04        1807525.       13956475.
      1806924.96     13956224.98
#Sta/Elev= 30
  4664.8  2109.6  4717.9 2107.46  4745.9 2107.36    4785 2105.94    4799 2104.59
  4874.5 2100.98  4880.1 2099.88  4910.8 2099.48  4919.2 2097.99  4941.6 2096.83
  4947.1  2094.9  4969.5 2090.45  4989.8  2088.8  4990.3  2088.3  5005.1  2088.8
  5032.8 2091.35  5086.4  2091.3  5108.6 2090.11  5139.5 2090.77  5174.1 2093.14
  5216.4 2094.59  5304.1 2094.25  5404.9 2095.72  5422.8 2097.79  5434.1    2101
  5452.5 2104.42  5466.1 2108.33  5529.5 2114.55  5606.4  2125.1  5650.3 2127.84
#Mann= 3 ,-1 , 0
  4664.8     .07       0  4989.8     .05       0  5005.1     .07       0
Bank Sta=4989.8,5005.1
XS Rating Curve= 0 ,0
Exp/Cntr=0.3,0.1

Type RM Length L Ch R = 1 ,52244   ,443,443,443
BEGIN DESCRIPTION:
Bear Creek 2 93.0
END DESCRIPTION:
XS GIS Cut Line= 3
      1808424.99     13956674.99        1807825.       13956125.
        1807625.     13955524.99
#Sta/Elev= 30
  4186.1 2125.39  4214.1 2123.74  4292.5 2116.28  4299.2 2116.54  4370.2 2110.62
  4419.5 2107.91  4568.1 2104.26    4627 2100.93  4660.6 2100.38  4759.2 2096.17
  4936.2 2092.04  4978.8  2087.8  5010.6 2086.97  5094.9 2088.33  5168.7 2087.65
  5210.9  2089.4  5245.4 2086.74  5245.9 2086.24  5260.7 2086.74  5274.1 2087.26
  5305.7 2091.05  5337.3 2092.33  5432.2 2092.14  5463.8 2093.28    5506 2096.75
  5537.6 2100.33  5548.2 2102.75  5579.8 2105.47  5611.4 2109.64  5632.5 2110.69
#Mann= 3 ,-1 , 0
  4186.1     .07       0  5245.4     .05       0  5260.7     .07       0
Bank Sta=5245.4,5260.7
XS Rating Curve= 0 ,0
Exp/Cntr=0.3,0.1

Type RM Length L Ch R = 1 ,51801   ,445,445,445
BEGIN DESCRIPTION:
Bear Creek 2 92.0
END DESCRIPTION:
XS GIS Cut Line= 3
      1808575.02     13956375.03        1808075.       13955775.
      1807925.02     13955425.04
#Sta/Elev= 30
  4223.8  2114.1  4309.1 2107.11  4436.7 2101.02    4519 2095.64    4572 2091.87
  4585.7 2091.78  4699.6 2090.04  4806.3 2090.32  4827.2 2091.45    4891 2090.28
  4905.3 2089.55  4919.6  2086.3  4933.9 2085.37  4948.2 2082.97  4962.6 2085.06
  4974.1 2082.83  4974.6 2082.33  4992.7 2082.83  5001.6 2085.79  5007.6 2085.79
  5019.4 2083.36  5059.3 2085.02  5090.1 2083.42  5124.5 2086.04  5218.8 2088.46
  5242.4 2090.71    5266 2095.43  5276.9 2098.99  5318.6 2105.54  5385.6 2109.77
#Mann= 5 ,-1 , 0
  4223.8     .07       0    4519      .1       0  4585.7     .07       0
  4974.1     .05       0  4992.7     .07       0
Bank Sta=4974.1,4992.7
XS Rating Curve= 0 ,0
Exp/Cntr=0.3,0.1

Type RM Length L Ch R = 1 ,51356   ,460,460,460
BEGIN DESCRIPTION:
Bear Creek 2 91.0
END DESCRIPTION:
XS GIS Cut Line= 3
        1808575.     13956174.99        1808425.       13955575.
        1808425.     13955374.95
#Sta/Elev= 30
  4390.1 2100.31  4413.3 2099.33  4431.3 2097.27  4515.9 2091.72  4518.4  2091.6
  4619.4 2088.87  4792.1    2088  4820.4 2085.69  4861.7 2084.22  4915.8 2084.11
  4949.3 2082.45  4967.3 2078.86  4968.3 2077.69  4968.8 2077.19  4986.9 2077.69
  4990.5 2079.06  4998.2 2080.22  5011.1 2081.18  5018.6 2083.81  5028.6 2085.92
  5048.6 2086.36  5088.6 2083.44  5108.6 2080.68  5118.6 2080.16  5138.6 2080.18
  5148.6 2081.26  5158.6  2085.4  5168.6 2097.25  5178.6 2101.25  5208.6 2103.88
#Mann= 5 ,-1 , 0
  4390.1     .07       0  4515.9      .1       0  4518.4     .07       0
  4968.3     .05       0  4986.9     .07       0
Bank Sta=4968.3,4986.9
XS Rating Curve= 0 ,0
Exp/Cntr=0.3,0.1

Type RM Length L Ch R = 1 ,50896   ,457,457,457
BEGIN DESCRIPTION:
Bear Creek 2 90.0
END DESCRIPTION:
XS GIS Cut Line= 3
        1809375.       13956025.        1808825.       13955425.
      1808674.98     13955274.98
#Sta/Elev= 30
  4185.4  2112.3  4270.2 2104.18  4326.9 2101.44  4440.4 2091.42  4461.3 2090.83
  4482.9 2088.25  4518.1 2086.19  4574.8 2084.44    4695 2083.39  4737.6 2079.05
  4758.5 2078.87  4765.9 2081.37  4786.9 2081.56  4808.5 2083.73  4843.6 2081.52
  4850.4 2082.08  4857.8    2080  4864.6 2080.28    4872 2078.03  4949.7 2079.04
  4986.6 2075.25  4987.1 2074.75  5005.2 2075.25  5013.5 2079.76  5027.6 2084.89
  5041.8 2087.72  5098.3 2092.98  5126.6 2093.79  5183.2 2098.62  5211.5 2099.63
#Mann= 3 ,-1 , 0
  4185.4     .07       0  4986.6     .05       0  5005.2     .07       0
Bank Sta=4986.6,5005.2
XS Rating Curve= 0 ,0
Exp/Cntr=0.3,0.1

Type RM Length L Ch R = 1 ,50439   ,482,482,482
BEGIN DESCRIPTION:
Bear Creek 2 89.0
END DESCRIPTION:
XS GIS Cut Line= 3
      1809475.01     13956025.01        1809225.       13955425.
      1808915.63     13954873.46
#Sta/Elev= 30
  4349.9 2114.13  4417.6 2110.37  4494.5 2102.11  4547.6 2098.18  4648.4 2083.75
  4739.9 2081.91  4837.4 2082.39  4879.1 2081.47  4961.5 2077.44  4967.4 2075.39
  4968.9 2072.46  4969.4 2071.96  4987.6 2072.46  4997.2  2075.1  5002.8  2075.1
  5007.9 2077.26  5035.3 2078.36  5045.5 2076.26  5072.9 2077.75  5088.9 2082.86
  5094.6 2082.77  5110.6 2085.34  5177.4 2087.26    5219 2086.79  5229.2 2088.29
  5250.5 2088.47  5337.7 2090.15  5456.3 2098.35  5492.9 2098.38  5632.3 2103.27
#Mann= 5 ,-1 , 0
  4349.9     .07       0  4968.9     .05       0  4987.6     .07       0
  5177.4    .035       0  5250.5     .07       0
Bank Sta=4968.9,4987.6
XS Rating Curve= 0 ,0
Exp/Cntr=0.3,0.1

Type RM Length L Ch R = 1 ,49957   ,442,442,442
BEGIN DESCRIPTION:
Bear Creek 2 88.0
END DESCRIPTION:
XS GIS Cut Line= 3
      1809974.99     13955574.99        1809675.       13955325.
      1809068.82     13954823.23
#Sta/Elev= 30
    4610 2109.71    4638 2109.51  4652.3 2106.58  4676.5 2094.67  4695.2  2083.9
  4716.1 2078.34  4799.5 2079.43  4844.3 2079.01  4894.4 2081.08  4950.4 2079.87
  4958.2    2079  4964.7 2075.32  4972.5 2075.65    4979 2068.95  4986.8 2068.55
  4987.9  2066.3  4988.4  2065.8  5006.6  2066.3  5036.3 2068.28  5050.7 2070.93
  5057.1 2076.73  5071.5 2081.18  5106.6 2083.77  5191.6 2084.22  5352.1 2086.29
  5511.7    2091  5554.6 2093.64  5575.5 2095.67  5634.8 2095.89  5787.4  2100.6
#Mann= 9 ,-1 , 0
    4610     .07       0  4676.5      .1       0  4799.5     .07       0
  4987.9     .05       0  5006.6     .07       0  5191.6    .035       0
  5352.1     .07       0  5554.6      .1       0  5634.8     .07       0
Bank Sta=4987.9,5006.6
XS Rating Curve= 0 ,0
Exp/Cntr=0.3,0.1

Type RM Length L Ch R = 1 ,49515   ,580,580,580
BEGIN DESCRIPTION:
Bear Creek 2 87.0
END DESCRIPTION:
XS GIS Cut Line= 3
        1810075.       13955475.        1810075.       13955275.
      1809475.02     13954675.02
#Sta/Elev= 30
  4796.1 2111.88  4846.1 2110.28  4876.1 2107.91  4886.1 2108.25  4916.1 2105.08
  4966.1  2086.3  4993.6 2074.03  4999.6 2074.03  5000.8 2071.39  5001.3 2070.89
  5019.6 2071.39  5052.7 2074.35  5095.1 2075.42  5109.2 2074.42  5123.4 2071.55
  5137.5 2071.82  5179.9 2075.87  5208.2 2077.14  5222.4  2076.4  5250.7 2077.04
  5278.9 2079.94  5349.7 2082.82  5420.4 2083.53  5434.5 2082.33  5519.4 2082.06
  5590.1 2082.58  5646.9 2084.31  5674.9 2084.61  5773.9 2088.43  5844.6 2094.13
#Mann= 4 ,-1 , 0
  4796.1     .07       0  5000.8     .05       0  5019.6     .07       0
  5646.9      .1       0
Bank Sta=5000.8,5019.6
XS Rating Curve= 0 ,0
Exp/Cntr=0.3,0.1
