HEC-RAS study Bear Creek 2.prj: Bear Creek 2 Base Level Engineering

--- Bear Creek 2.g01 (geometry) --- (continued)

Type RM Length L Ch R = 1 ,48935   ,577,577,577
BEGIN DESCRIPTION:
Bear Creek 2 86.0
END DESCRIPTION:
XS GIS Cut Line= 3
      1810625.03     13954574.98        1810275.       13954775.
      1809474.99       13954625.
#Sta/Elev= 30
  4604.6 2102.53  4695.5 2096.65  4801.2 2090.87  4823.5  2089.2  4832.8 2087.06
  4838.6  2087.8  4854.4  2078.8  4860.2 2079.86    4876 2071.01  4897.6 2070.72
  4904.1 2069.11  4919.2 2069.04    4935 2071.07  4961.7  2068.8  4962.2  2068.3
  4983.3  2068.8  5017.9 2071.95  5039.1 2071.78  5099.3  2075.4  5139.2 2076.37
  5190.9 2076.86  5262.1 2074.63    5307 2077.07  5333.3 2079.59  5412.2 2080.72
  5482.4 2079.75  5587.7 2081.71  5709.8 2086.62    5781 2093.66  5821.7    2096
#Mann= 5 ,-1 , 0
  4604.6      .1       0  4695.5     .07       0  4961.7     .05       0
  4983.3     .07       0  5482.4      .1       0
Bank Sta=4961.7,4983.3
XS Rating Curve= 0 ,0
Exp/Cntr=0.3,0.1

Type RM Length L Ch R = 1 ,48358   ,564,564,564
BEGIN DESCRIPTION:
Bear Creek 2 85.0
END DESCRIPTION:
XS GIS Cut Line= 3
        1810675.       13954175.        1810275.       13954225.
      1809475.02       13954225.
#Sta/Elev= 30
  4596.5 2125.09  4687.2 2122.77  4714.9 2118.98  4747.7 2117.28  4838.4 2108.24
  4868.6 2099.81  4876.2    2095  4881.2 2093.35  4888.8 2085.11  4898.8 2078.17
    4920 2070.19  4929.1 2067.67  4961.8 2070.67  4969.4 2070.53  4977.3 2068.22
  4986.2 2065.32  4986.7 2064.82  5007.9 2065.32  5029.6 2065.44  5049.6 2069.67
  5089.6 2069.94  5109.6 2068.44  5149.6 2073.28  5169.6 2073.99  5239.6 2073.51
  5259.6 2074.82  5299.6  2072.5  5389.6 2077.67  5579.6 2080.51  5799.6 2095.29
#Mann= 5 ,-1 , 0
  4596.5      .1       0    4920     .07       0  4977.3      .1       0
  4986.2     .05       0  5007.9      .1       0
Bank Sta=4986.2,5007.9
XS Rating Curve= 0 ,0
Exp/Cntr=0.3,0.1

Type RM Length L Ch R = 1 ,47794   ,587,587,587
BEGIN DESCRIPTION:
Bear Creek 2 84.0
END DESCRIPTION:
XS GIS Cut Line= 3
      1810575.02     13953624.99        1810175.       13953725.
        1809475.       13954175.
#Sta/Elev= 30
  4591.9 2130.55  4664.1 2124.26  4725.9 2115.07  4767.2 2101.66  4839.3 2073.67
  4857.3  2069.8  4939.8 2071.12  4952.7 2070.72  4973.3 2066.57  4986.2 2066.17
  5001.7 2068.01  5039.9 2067.43  5069.3 2068.76  5099.3 2067.43  5120.8 2070.46
  5199.4 2071.11  5265.8 2068.69  5303.5 2065.03    5304 2064.53  5325.2 2065.03
  5329.5 2069.09    5346 2074.33  5553.4  2078.9  5620.2 2082.37  5662.4 2083.97
  5756.2 2090.65  5771.3    2093  5792.5 2092.41  5807.7 2094.02  5836.4 2094.49
#Mann= 5 ,-1 , 0
  4591.9      .1       0  5303.5     .05       0  5325.2      .1       0
    5346     .07       0  5620.2      .1       0
Bank Sta=5303.5,5325.2
XS Rating Curve= 0 ,0
Exp/Cntr=0.3,0.1

Type RM Length L Ch R = 1 ,47207   ,535,535,535
BEGIN DESCRIPTION:
Bear Creek 2 83.0
END DESCRIPTION:
XS GIS Cut Line= 3
      1810424.98     13953374.99        1810075.       13953175.
      1809274.97     13953825.02
#Sta/Elev= 30
  4596.8 2121.53  4771.7 2113.42  4787.5 2108.77  4809.1 2106.32    4825 2100.86
  4830.7 2101.08  4846.6  2094.1  4852.3 2094.33  4861.7 2090.92  4868.2  2086.9
  4889.8 2084.07  4905.6 2074.44  4911.3 2075.03  4927.2 2066.32  4970.4 2064.47
    4992 2061.37    5071 2067.68  5196.9 2066.92  5239.1 2065.56  5251.9  2060.6
  5252.4  2060.1  5273.6  2060.6  5283.6 2064.22  5328.3 2067.42  5454.6 2074.81
  5654.3 2080.58  5796.5 2082.52  5874.8 2086.02  5959.6 2093.45  6030.7 2096.73
#Mann= 6 ,-1 , 0
  4596.8      .1       0  5196.9     .07       0  5239.1      .1       0
  5251.9     .05       0  5273.6      .1       0  5328.3     .07       0
Bank Sta=5251.9,5273.6
XS Rating Curve= 0 ,0
Exp/Cntr=0.3,0.1

Type RM Length L Ch R = 1 ,46672   ,581,581,581
BEGIN DESCRIPTION:
Bear Creek 2 82.0
END DESCRIPTION:
XS GIS Cut Line= 4
        1810275.       13952925.       1810166.6      13952751.5
        1809925.       13952725.      1808909.63      13952855.9
#Sta/Elev= 30
  4556.9 2104.93  4651.2  2100.3  4686.6 2092.69  4710.2 2091.05  4737.9  2086.7
  4764.8 2085.24  4776.7  2083.1  4793.3 2074.85  4813.4 2068.84  4833.5 2065.99
    4914 2064.38  4983.4  2059.5  4983.9    2059  5005.6  2059.5  5085.2 2062.73
  5105.4  2066.5  5115.4 2066.76  5195.6 2066.46  5216.3 2062.48    5234 2062.78
  5256.6 2062.63  5296.9 2067.44  5387.7  2072.4  5458.2 2074.96    5549 2073.16
  5569.2 2075.85  5690.2 2078.99  5751.6 2083.23  5932.1 2090.13  6028.3  2096.3
#Mann= 4 ,-1 , 0
  4556.9      .1       0  4983.4     .05       0  5005.6      .1       0
    5234     .07       0
Bank Sta=4983.4,5005.6
XS Rating Curve= 0 ,0
Exp/Cntr=0.3,0.1

Type RM Length L Ch R = 1 ,46091   ,530,530,530
BEGIN DESCRIPTION:
Bear Creek 2 81.0
END DESCRIPTION:
XS GIS Cut Line= 3
      1810374.98       13952275.        1809925.       13952175.
        1809175.       13951725.
#Sta/Elev= 30
    4544  2098.1  4657.3 2086.04  4666.9  2086.3  4677.2 2083.39  4718.1 2080.06
  4759.1 2074.21  4810.3 2071.08  4851.3 2062.45  4879.5 2061.17  4937.1 2060.39
  4953.7 2055.57  4963.1 2055.56  4963.6 2055.06  4985.4 2055.56  5002.4 2058.09
  5089.2 2060.79  5129.4 2063.04  5261.5 2063.62  5354.8 2059.69  5479.2 2063.11
  5565.5 2063.29  5583.3 2063.62  5611.4 2065.81  5638.6 2070.87  5681.4 2088.73
  5696.9    2092  5739.7 2105.73    5796 2115.78  5844.8 2120.57  5879.6 2122.69
#Mann= 10 ,-1 , 0
    4544      .1       0  4657.3     .07       0  4879.5      .1       0
  4963.1     .05       0  4985.4      .1       0  5089.2     .07       0
  5565.5      .1       0  5583.3     .07       0    5796      .1       0
  5844.8     .07       0
Bank Sta=4963.1,4985.4
XS Rating Curve= 0 ,0
Exp/Cntr=0.3,0.1

Type RM Length L Ch R = 1 ,45561   ,534,534,534
BEGIN DESCRIPTION:
Bear Creek 2 80.0
END DESCRIPTION:
XS GIS Cut Line= 3
      1810575.03     13952075.01        1809775.       13951725.
      1809274.96     13951574.99
#Sta/Elev= 30
  4132.8  2108.4  4293.1 2094.45  4345.3 2091.36  4401.6 2084.49  4496.5 2073.21
  4569.4 2070.56  4733.2 2065.87  4840.4 2059.22  4929.6 2058.55  4973.1 2056.83
  4973.6 2056.33  4995.4 2056.83  5037.4 2059.35  5093.9  2058.2  5146.7 2061.13
  5187.7 2059.46  5214.8  2059.4  5236.6 2061.56  5325.1 2062.28    5341 2063.57
    5361 2068.28  5368.8 2072.76  5374.1 2073.75  5381.9 2078.81  5407.1 2090.67
  5413.2 2095.33  5440.2 2108.52  5465.4 2114.63  5473.2 2117.75  5528.1 2122.96
#Mann= 8 ,-1 , 0
  4132.8      .1       0  4401.6     .07       0  4569.4      .1       0
  4973.1     .05       0  4995.4      .1       0  5146.7     .07       0
  5187.7      .1       0  5325.1     .07       0
Bank Sta=4973.1,4995.4
XS Rating Curve= 0 ,0
Exp/Cntr=0.3,0.1

Type RM Length L Ch R = 1 ,45027   ,544,544,544
BEGIN DESCRIPTION:
Bear Creek 2 79.0
END DESCRIPTION:
XS GIS Cut Line= 3
      1810575.01     13951925.01        1809775.       13951225.
        1809325.       13951275.
#Sta/Elev= 30
  3932.1 2103.71  3960.1 2102.13  3996.2  2097.5  4031.3 2096.35  4059.8 2092.19
  4105.9  2088.6    4215 2074.89  4229.7 2072.98  4342.4 2067.45  4710.9 2060.03
  4775.4 2058.77  4803.9  2056.7  4853.2  2056.8  4895.9 2058.82  4952.9 2055.76
  4979.2 2055.89  4991.8 2055.43  4993.9 2053.94  4994.4 2053.44  5016.5 2053.94
  5065.6 2057.14  5115.9 2054.74  5166.2 2059.83  5216.5  2061.6  5232.3 2064.04
  5233.4 2064.31  5246.7 2068.02  5337.2 2103.66  5397.6  2117.2  5447.9 2121.14
#Mann= 10 ,-1 , 0
  3932.1      .1       0  4105.9     .07       0    4215    .035       0
  4342.4     .07       0  4710.9      .1       0  4979.2     .07       0
  4993.9     .05       0  5016.5     .07       0  5232.3      .1       0
  5233.4     .07       0
Bank Sta=4993.9,5016.5
XS Rating Curve= 0 ,0
Exp/Cntr=0.3,0.1

Type RM Length L Ch R = 1 ,44483   ,534,534,534
BEGIN DESCRIPTION:
Bear Creek 2 78.0
END DESCRIPTION:
XS GIS Cut Line= 3
      1810774.99     13951574.99        1809975.       13950775.
      1809624.98     13950574.99
#Sta/Elev= 30
    3863  2094.7  4004.4 2086.19  4117.5 2071.41    4192 2066.41  4287.3 2062.39
  4391.7 2061.35  4421.1 2061.26    4559 2061.12  4654.9 2054.66  4777.1 2058.21
  4881.2 2055.69  4923.6 2051.91  4980.2 2051.97  4990.8 2049.63    4991 2048.01
  4991.5 2047.51  5013.6 2048.01  5080.7 2055.61  5110.3 2071.64  5120.3 2073.85
  5126.1 2078.78  5141.9  2083.7  5147.7  2088.7  5163.5 2093.48  5169.3 2098.59
  5185.1 2103.88  5190.9 2108.65  5228.3 2120.08  5249.9 2124.15  5397.5 2126.84
#Mann= 8 ,-1 , 0
    3863     .07       0    4192    .035       0  4391.7     .07       0
  4421.1      .1       0    4559     .07       0  4777.1      .1       0
    4991     .05       0  5013.6      .1       0
Bank Sta=4991,5013.6
XS Rating Curve= 0 ,0
Exp/Cntr=0.3,0.1

Type RM Length L Ch R = 1 ,43949   ,558,558,558
BEGIN DESCRIPTION:
Bear Creek 2 77.0
END DESCRIPTION:
XS GIS Cut Line= 3
      1810875.02     13951375.03        1810375.       13950575.
      1810175.02     13950225.04
#Sta/Elev= 30
  4046.4 2084.94  4199.7 2076.92  4265.1  2069.1  4337.9 2065.36  4553.5 2060.43
  4765.8 2058.35  4903.2 2050.71  4943.6 2051.01  4997.8 2049.51  5062.5 2051.15
  5094.4 2048.67  5094.9 2048.17  5117.1 2048.67  5121.6 2051.45  5137.4 2055.68
  5164.8 2070.88    5218 2087.84  5223.8 2091.04  5239.6 2094.58  5245.4 2098.03
    5267 2104.59  5277.1 2105.21  5282.8 2107.92  5304.4 2109.51  5320.2  2105.9
    5326  2106.9  5341.8 2101.79  5363.4 2100.17  5379.3 2095.29  5392.9 2093.83
#Mann= 6 ,-1 , 0
  4046.4     .07       0  4265.1    .035       0  4337.9     .07       0
  4943.6      .1       0  5094.4     .05       0  5117.1      .1       0
Bank Sta=5094.4,5117.1
XS Rating Curve= 0 ,0
Exp/Cntr=0.3,0.1

Type RM Length L Ch R = 1 ,43391   ,566,566,566
BEGIN DESCRIPTION:
Bear Creek 2 76.0
END DESCRIPTION:
XS GIS Cut Line= 3
      1810987.71     13951340.85        1810825.       13950275.
      1811075.01     13949474.96
#Sta/Elev= 30
  3926.3 2083.84  4010.4 2079.62  4114.7 2074.58  4185.1 2069.02  4255.9 2066.22
  4427.9    2065  4573.1  2060.4  4599.9 2057.51  4634.3 2056.68  4736.1 2054.46
  4822.4 2049.55  4893.2 2049.94  4990.6 2046.33  4991.1 2045.83  5013.3 2046.33
  5035.9 2048.41  5058.5  2047.5  5085.7 2050.81    5173 2052.32  5193.6 2051.79
    5214 2048.08    5284 2050.59  5507.4 2053.07  5593.8 2056.77  5621.1 2061.02
  5626.3 2060.31  5691.3 2068.24    5729 2071.21  5779.8 2078.62  5842.7 2091.02
#Mann= 9 ,-1 , 0
  3926.3      .1       0  4010.4     .07       0  4573.1      .1       0
  4634.3     .07       0  4736.1      .1       0  4990.6     .05       0
  5013.3      .1       0    5173     .07       0    5284      .1       0
Bank Sta=4990.6,5013.3
XS Rating Curve= 0 ,0
Exp/Cntr=0.3,0.1

Type RM Length L Ch R = 1 ,42825   ,565,565,565
BEGIN DESCRIPTION:
Bear Creek 2 75.0
END DESCRIPTION:
XS GIS Cut Line= 3
      1811775.01     13950875.02        1811275.       13950075.
      1811174.99     13949324.95
#Sta/Elev= 30
  4056.6 2086.32  4237.6 2074.57  4312.4 2067.92  4405.1 2062.51  4541.6 2059.64
  4705.4 2053.41  4834.7 2051.49  4870.3    2051  4905.7 2047.62  4986.5 2044.36
  5030.3 2046.51  5058.5 2044.08    5059 2043.58  5082.8 2044.08  5109.7  2047.5
  5153.4 2048.46  5211.9 2044.59  5232.1 2047.01  5255.9 2047.42  5282.5 2049.51
  5332.9 2049.83  5417.4 2056.68  5490.6 2068.88  5495.6 2068.47  5524.6 2074.26
  5615.4 2094.49  5635.6 2099.64  5641.9 2102.67    5715 2113.34  5756.7 2116.76
#Mann= 9 ,-1 , 0
  4056.6      .1       0  4312.4     .07       0  4541.6      .1       0
  4705.4     .07       0  4834.7      .1       0  5058.5     .05       0
  5082.8      .1       0  5153.4     .07       0  5255.9      .1       0
Bank Sta=5058.5,5082.8
XS Rating Curve= 0 ,0
Exp/Cntr=0.3,0.1

Type RM Length L Ch R = 1 ,42260   ,517,517,517
BEGIN DESCRIPTION:
Bear Creek 2 74.0
END DESCRIPTION:
XS GIS Cut Line= 3
        1811875.       13951075.        1811675.       13949675.
        1811525.     13949275.01
#Sta/Elev= 30
  3585.8 2104.73  3646.4 2102.01  3764.8 2090.61  3959.6 2077.82  4051.1 2070.01
  4191.9 2062.05  4452.8 2054.95  4518.8 2052.56    4628 2050.25  4684.9 2048.39
  4808.6 2048.28    4899 2047.78  4939.4 2045.09  4969.7 2039.88  4985.3 2038.99
  4985.8 2038.49  5009.7 2038.99  5040.1 2044.02  5100.6 2042.74  5130.8  2044.8
  5180.7 2043.95  5192.3 2050.78  5210.9 2057.27  5241.2 2066.75  5271.5 2072.56
  5320.4  2087.8  5326.6 2091.27  5363.1  2101.4  5395.2 2108.27  5427.2 2111.02
#Mann= 10 ,-1 , 0
  3585.8     .07       0  3764.8      .1       0  4051.1     .07       0
  4452.8      .1       0  4518.8     .07       0    4628      .1       0
  4684.9     .07       0  4808.6      .1       0  4985.3     .05       0
  5009.7      .1       0
Bank Sta=4985.3,5009.7
XS Rating Curve= 0 ,0
Exp/Cntr=0.3,0.1

Type RM Length L Ch R = 1 ,41743   ,546,546,546
BEGIN DESCRIPTION:
Bear Creek 2 73.0
END DESCRIPTION:
XS GIS Cut Line= 3
        1811925.     13950925.01        1812025.       13949375.
      1811675.04     13949175.02
#Sta/Elev= 30
  3441.3 2096.92  3492.9  2091.6  3571.6 2085.05  3762.7 2074.33  4012.5 2059.68
  4185.9 2054.44  4252.5 2052.77  4542.8 2048.23  4663.9 2044.75    4754 2044.72
  4774.1 2041.43  4884.3 2045.22  4934.4 2044.49  4964.5 2040.98  5002.5 2040.07
  5017.6 2035.84  5018.1 2035.34    5042 2035.84  5045.6  2037.9  5083.1 2038.26
  5088.8 2044.03  5104.7 2047.88  5110.4 2054.47  5120.5  2056.1  5126.3 2061.73
  5132.7 2064.73  5163.7  2075.7  5169.5  2080.5  5191.1 2085.54  5397.6 2103.82
#Mann= 8 ,-1 , 0
  3441.3     .07       0  3492.9      .1       0  3762.7     .07       0
  4185.9      .1       0  4252.5     .07       0  4542.8      .1       0
  5017.6     .05       0    5042      .1       0
Bank Sta=5017.6,5042
XS Rating Curve= 0 ,0
Exp/Cntr=0.3,0.1

Type RM Length L Ch R = 1 ,41197   ,553,553,553
BEGIN DESCRIPTION:
Bear Creek 2 72.0
END DESCRIPTION:
XS GIS Cut Line= 3
        1811975.     13950974.99        1812525.       13949425.
        1812225.     13948975.01
#Sta/Elev= 30
  3345.5 2101.05  3391.8 2097.83  3430.4 2093.06  3485.2 2089.58  3610.8 2082.38
    3753 2077.77  3950.3 2065.68  4049.7 2062.93  4137.3 2058.21    4435 2049.26
    4640 2048.02  4809.8 2041.91  4918.3 2041.85  4958.3 2039.37  4987.5 2035.24
  5003.7 2034.88  5026.2 2036.71  5039.8    2035  5048.8 2035.77    5050 2034.31
  5050.5 2033.81  5074.6 2034.31  5084.8 2039.56  5090.8 2038.58  5098.3    2045
  5105.9 2046.72  5201.2    2050    5229 2051.67  5445.4 2057.32    5531 2061.61
#Mann= 7 ,-1 , 0
  3345.5     .07       0  3485.2      .1       0    3753     .07       0
  4137.3      .1       0    5050     .05       0  5074.6      .1       0
  5201.2     .07       0
Bank Sta=5050,5074.6
XS Rating Curve= 0 ,0
Exp/Cntr=0.3,0.1

Type RM Length L Ch R = 1 ,40644   ,534,534,534
BEGIN DESCRIPTION:
Bear Creek 2 71.0
END DESCRIPTION:
XS GIS Cut Line= 3
      1812616.21     13950298.64      1813064.28     13949506.78
      1812375.02     13948775.02
#Sta/Elev= 30
  4173.4 2055.75  4269.5 2051.88  4475.7 2048.46  4704.7 2045.42  4740.6 2041.28
  4808.1 2040.87  4850.5 2040.69  4856.2 2038.48  4866.4 2040.79    4888 2040.52
  4958.9 2037.63  4974.6 2036.43  4981.9 2033.74  4983.9 2030.75  4984.4 2030.25
  5008.5 2030.75  5008.7 2030.85  5012.1 2032.47  5098.3 2039.29  5303.4 2041.94
  5381.1 2039.98  5419.5 2040.78  5515.4  2043.5  5635.6 2049.59  5678.1 2048.16
  5699.5 2045.62    5827 2050.94  5925.7  2050.7  5961.3  2054.8  6088.5    2059
#Mann= 7 ,-1 , 0
  4173.4     .07       0  4475.7      .1       0  4808.1     .07       0
  4983.9     .05       0  5008.5     .07       0  5008.7      .1       0
  5419.5     .07       0
Bank Sta=4983.9,5008.5
XS Rating Curve= 0 ,0
Exp/Cntr=0.3,0.1

Type RM Length L Ch R = 1 ,40110   ,532,532,532
BEGIN DESCRIPTION:
Bear Creek 2 70.0
END DESCRIPTION:
XS GIS Cut Line= 3
      1813675.01     13949625.01        1813375.       13949325.
      1812774.98     13948874.98
#Sta/Elev= 30
  4580.5 2111.07  4594.6 2110.34  4608.8 2107.66  4736.1 2077.44  4778.5 2070.58
    4828 2065.35  4891.6 2055.33  4919.9 2052.18  4948.2 2035.58  4962.3 2030.85
  4976.5 2028.81  4977.8 2026.59  4978.3 2026.09  5003.5 2026.59  5007.9 2027.57
  5012.1 2030.65  5047.5 2037.91  5082.9 2039.81  5191.2 2041.52  5226.6 2041.31
  5241.2 2038.78  5254.8 2038.58  5291.2 2040.64  5326.6 2039.92  5347.5 2041.03
  5412.1 2038.79  5447.5 2042.95  5518.3 2047.13  5595.7 2049.01  5754.8 2051.61
#Mann= 4 ,-1 , 0
  4580.5      .1       0  4977.8     .05       0  5003.5      .1       0
  5595.7     .07       0
Bank Sta=4977.8,5003.5
XS Rating Curve= 0 ,0
Exp/Cntr=0.3,0.1

Type RM Length L Ch R = 1 ,39578   ,614,614,614
BEGIN DESCRIPTION:
Bear Creek 2 69.0
END DESCRIPTION:
XS GIS Cut Line= 4
        1813825.     13949425.02      1813784.55     13949020.55
      1813665.79     13948877.22      1812175.04     13948225.02
#Sta/Elev= 30
  4519.3 2090.53  4567.1 2080.68  4599.7 2076.69  4873.6 2055.83  4925.8 2044.21
  4929.7 2040.69  4934.1  2039.2  4950.5 2033.49    4952  2030.1  4952.5  2029.6
  4977.8  2030.1  5057.3 2032.79  5071.7  2031.2  5115.1 2031.43  5129.6 2034.75
  5158.4 2037.75  5243.8  2038.3  5265.6 2037.55  5287.4 2033.84  5320.2 2036.64
  5426.6 2040.65  5576.7 2040.78  5669.5 2043.99  5891.5 2047.55  6040.6 2052.55
  6229.6 2053.51  6578.9 2060.58  6640.9 2064.58  6701.3 2074.71  6739.1 2077.39
#Mann= 6 ,-1 , 0
  4519.3      .1       0  4934.1     .07       0    4952     .05       0
  4977.8     .07       0  5576.7      .1       0  5891.5     .07       0
Bank Sta=4952,4977.8
XS Rating Curve= 0 ,0
Exp/Cntr=0.3,0.1

Type RM Length L Ch R = 1 ,38964   ,524,524,524
BEGIN DESCRIPTION:
Bear Creek 2 68.0
END DESCRIPTION:
XS GIS Cut Line= 3
      1814424.96     13948624.99        1813975.       13948475.
      1813224.99     13947974.99
#Sta/Elev= 30
  4525.3 2052.75  4539.8 2052.51  4642.5 2049.82  4662.3 2047.86  4704.5 2037.37
  4736.1 2033.58  4746.6 2034.15  4757.2 2033.25  4820.4 2032.99  4841.5 2032.52
    4852  2031.1  4925.8 2030.52    4968 2028.54  4978.5 2028.64  4989.1 2030.13
  4993.6 2027.13  4994.1 2026.63  5020.6 2027.13  5022.1 2028.79  5035.7 2029.25
  5043.2 2031.26  5071.7 2030.96  5094.2 2036.69  5130.3 2039.47  5232.7 2038.92
  5382.7  2042.3  5511.1 2043.52  5749.3 2050.46  5857.4 2056.31    5901 2056.88
#Mann= 7 ,-1 , 0
  4525.3      .1       0  4539.8     .07       0  4642.5      .1       0
  4993.6     .05       0  5020.6      .1       0  5232.7      .1       0
  5511.1     .07       0
Bank Sta=4993.6,5020.6
XS Rating Curve= 0 ,0
Exp/Cntr=0.3,0.1

Type RM Length L Ch R = 1 ,38440   ,538,538,538
BEGIN DESCRIPTION:
Bear Creek 2 67.0
END DESCRIPTION:
XS GIS Cut Line= 3
      1814475.01     13948275.01        1814125.       13948025.
      1813475.04     13947625.02
#Sta/Elev= 30
  4574.6  2053.7  4602.9 2053.27  4623.8 2051.61  4653.3 2041.14  4666.8 2035.21
  4674.2  2030.3  4682.8 2026.32  4696.3 2024.83  4696.8 2024.33  4723.3 2024.83
  4724.5 2026.78  4746.7  2030.1  4854.8  2032.1  4888.5 2031.35  4918.7 2031.12
  4941.4 2027.97  4976.5 2028.99  4991.2 2026.68  5007.2 2026.77  5012.4 2028.47
  5033.7 2028.14  5076.3 2029.77  5107.1 2034.41  5183.8 2038.24  5265.6 2040.33
  5372.8 2040.26  5470.4 2041.02  5543.8 2043.02  5723.5 2055.29  5767.9 2056.71
#Mann= 8 ,-1 , 0
  4574.6      .1       0  4696.3     .05       0  4723.3      .1       0
  4888.5     .07       0  4941.4      .1       0  5007.2     .07       0
  5183.8      .1       0  5372.8     .07       0
Bank Sta=4696.3,4723.3
XS Rating Curve= 0 ,0
Exp/Cntr=0.3,0.1

Type RM Length L Ch R = 1 ,37902   ,512,512,512
BEGIN DESCRIPTION:
Bear Creek 2 66.0
END DESCRIPTION:
XS GIS Cut Line= 3
      1814675.03     13947875.03        1814375.       13947575.
      1813675.03     13947175.02
#Sta/Elev= 30
  4575.9 2051.93  4646.8 2047.02  4759.8 2037.37  4788.1 2031.27  4802.2 2025.49
  4816.4 2021.94  4858.8 2023.06  4859.4 2021.88  4859.9 2021.38  4886.4 2021.88
  4887.1 2027.78  4943.6  2026.8  4986.1 2029.42  4996.7 2026.88  5003.1 2026.88
  5008.1 2023.93  5013.9 2023.43  5072.9 2027.39  5103.9  2028.2  5110.3 2026.94
  5196.7  2027.4  5234.2 2029.08  5265.1 2032.58  5293.2 2033.18  5322.7 2035.87
    5417 2037.78  5622.2 2046.28  5702.8 2055.16  5755.3 2058.49  5806.4 2059.48
#Mann= 4 ,-1 , 0
  4575.9      .1       0  4646.8     .07       0  4859.4     .05       0
  4886.4     .07       0
Bank Sta=4859.4,4886.4
XS Rating Curve= 0 ,0
Exp/Cntr=0.3,0.1

Type RM Length L Ch R = 1 ,37390   ,529,529,529
BEGIN DESCRIPTION:
Bear Creek 2 65.0
END DESCRIPTION:
XS GIS Cut Line= 3
      1814975.01     13947775.02        1814625.       13947175.
      1814274.97     13946974.98
#Sta/Elev= 30
  4306.3 2055.31  4351.4 2052.94  4394.4 2048.63  4468.4 2045.06  4496.1 2045.17
    4549 2041.04  4607.3 2040.91  4709.5 2038.37    4817 2034.48  4912.9 2029.54
  4934.4 2029.45  4965.8 2026.25  4971.6 2022.92  4977.8 2021.78  4984.5 2018.96
    4985 2018.46  5011.6 2018.96  5052.1 2020.75  5081.6 2020.47  5104.6  2022.4
  5111.1 2024.84  5148.5 2025.61  5197.5  2020.7  5213.3 2022.07  5229.1 2025.21
  5234.9 2028.63  5256.5 2036.09  5278.1 2040.14  5315.5 2043.54  5404.1 2045.47
#Mann= 3 ,-1 , 0
  4306.3     .07       0  4984.5     .05       0  5011.6     .07       0
Bank Sta=4984.5,5011.6
XS Rating Curve= 0 ,0
Exp/Cntr=0.3,0.1

Type RM Length L Ch R = 1 ,36861   ,589,589,589
BEGIN DESCRIPTION:
Bear Creek 2 64.0
END DESCRIPTION:
XS GIS Cut Line= 3
      1815225.03     13946975.01        1814675.       13946725.
        1814275.       13946675.
#Sta/Elev= 30
  4400.1 2043.26  4455.1 2040.94  4513.5 2035.14  4561.2 2032.59  4586.9 2030.85
  4627.5 2029.96    4633 2029.24  4725.3 2027.06  4740.7 2026.08  4776.9 2022.06
  4846.1  2022.5  4874.7 2021.38  4892.2 2022.91  4905.4 2022.76  4920.8 2021.49
  4960.3 2020.19  4966.9 2018.88  4968.6 2017.38  4969.1 2016.88    4996 2017.38
  5001.5 2019.81  5034.5 2021.28  5054.7 2023.94  5122.7 2027.43  5185.7 2037.39
  5207.2 2039.13    5226 2040.43  5256.2 2040.81  5357.1 2044.47  5407.4 2045.49
#Mann= 7 ,-1 , 0
  4400.1     .07       0  4513.5      .1       0  4561.2     .07       0
  4968.6     .05       0    4996     .07       0  5207.2      .1       0
  5357.1     .07       0
Bank Sta=4968.6,4996
XS Rating Curve= 0 ,0
Exp/Cntr=0.3,0.1

Type RM Length L Ch R = 1 ,36272   ,520,520,520
BEGIN DESCRIPTION:
Bear Creek 2 63.0
END DESCRIPTION:
XS GIS Cut Line= 3
      1815425.02     13946575.01        1815075.       13946325.
      1814874.98     13945824.96
#Sta/Elev= 30
  4563.1 2041.98    4600 2040.88  4635.6 2038.29    4686 2031.97  4706.9 2027.59
  4721.6 2025.82  4821.2 2021.05  4893.7 2019.16  4899.8 2017.62  4907.3 2017.11
  4957.3 2015.26  4957.8 2014.76  4984.9 2015.26  4985.9 2016.67  4995.9 2016.19
  5014.8 2018.13  5025.5 2017.84  5037.7 2015.91  5047.1 2016.34  5086.1 2024.72
  5100.9 2026.28  5145.4 2029.03  5218.1 2030.94  5262.5 2034.76    5284  2037.9
  5294.8 2038.33  5360.8 2048.13  5445.6  2057.1  5516.9  2065.9  5531.8 2066.43
#Mann= 4 ,-1 , 0
  4563.1     .07       0  4907.3      .1       0  4957.3     .05       0
  4984.9     .07       0
Bank Sta=4957.3,4984.9
XS Rating Curve= 0 ,0
Exp/Cntr=0.3,0.1

Type RM Length L Ch R = 1 ,35752   ,445,445,445
BEGIN DESCRIPTION:
Bear Creek 2 62.0
END DESCRIPTION:
XS GIS Cut Line= 3
        1815575.       13946375.        1815375.       13946025.
      1815074.98     13945724.98
#Sta/Elev= 30
  4596.9 2038.75  4642.3 2038.38  4700.6 2036.46    4707 2036.88  4803.5    2033
  4825.1 2031.08  4830.8 2028.71  4846.7 2026.87  4852.4 2024.51  4861.8 2023.71
    4874 2020.34  4899.5 2016.01  4905.7 2015.58  4911.5 2014.08  4927.3 2015.29
  4942.4 2013.68    5000 2013.15  5000.4 2012.39  5000.9 2011.89    5028 2012.39
  5028.3 2013.09  5050.4 2015.36  5106.1 2019.96  5127.3 2023.03  5169.7 2026.44
  5254.6 2040.53  5282.9 2047.16  5325.3 2052.73    5396 2060.59  5424.3 2062.96
#Mann= 5 ,-1 , 0
  4596.9     .07       0  4899.5      .1       0  5000.4     .05       0
    5028      .1       0  5050.4     .07       0
Bank Sta=5000.4,5028
XS Rating Curve= 0 ,0
Exp/Cntr=0.3,0.1

Type RM Length L Ch R = 1 ,35307   ,636,636,636
BEGIN DESCRIPTION:
Bear Creek 2 61.0
END DESCRIPTION:
XS GIS Cut Line= 4
        1815725.     13946475.03      1815765.32     13945829.95
      1815642.49     13945641.87      1815374.99       13945575.
#Sta/Elev= 30
  4248.6 2036.98  4338.8 2035.26  4519.2 2033.44  4651.9 2029.53  4699.5 2029.15
  4739.6 2027.87  4839.8  2023.3  4869.8 2020.86  4920.9 2013.65    4936 2012.69
  4957.1 2013.54  4994.5 2011.01    4995 2010.51  5022.1 2011.01  5044.2 2016.15
  5050.6 2016.61  5071.6    2016  5101.9 2012.59  5119.1 2013.24  5137.6 2015.67
  5158.2 2019.71  5165.9 2022.06  5171.1 2025.77  5178.8 2026.97  5212.3 2037.78
  5230.4 2042.04  5253.6 2045.21  5271.6 2046.75  5343.8  2049.3  5395.3 2052.36
#Mann= 4 ,-1 , 0
  4248.6      .1       0  4994.5     .05       0  5022.1      .1       0
  5119.1     .07       0
Bank Sta=4994.5,5022.1
XS Rating Curve= 0 ,0
Exp/Cntr=0.3,0.1

Type RM Length L Ch R = 1 ,34671   ,565,565,565
BEGIN DESCRIPTION:
Bear Creek 2 60.0
END DESCRIPTION:
XS GIS Cut Line= 3
        1816575.     13946224.99        1816225.       13945425.
      1815825.01     13944625.03
#Sta/Elev= 30
  4130.9 2045.33  4267.7 2035.74  4360.1 2033.36  4600.2 2021.55  4726.9 2018.53
  4791.6 2014.28  4843.9 2014.49  4851.3 2039.02  4861.8 2013.01  4960.4 2009.46
  4968.4 2007.89  4968.9 2007.39  4996.2 2007.89  5040.4 2010.67  5079.6 2021.47
  5107.5  2026.4  5129.9 2027.92  5169.1 2027.71  5219.3  2028.2  5353.5 2023.22
  5370.3 2021.51  5375.8 2022.33  5392.6 2017.66  5412.2  2018.1  5591.8 2022.67
  5688.5 2024.95  5733.6  2027.3  5750.4 2030.05  5817.5 2035.75  5898.5 2038.94
#Mann= 8 ,-1 , 0
  4130.9     .07       0  4726.9      .1       0  4968.4     .05       0
  4996.2      .1       0  5169.1     .07       0  5412.2      .1       0
  5591.8     .07       0  5688.5      .1       0
Bank Sta=4968.4,4996.2
XS Rating Curve= 0 ,0
Exp/Cntr=0.3,0.1

Type RM Length L Ch R = 1 ,34106   ,540,540,540
BEGIN DESCRIPTION:
Bear Creek 2 59.0
END DESCRIPTION:
XS GIS Cut Line= 3
      1817224.97     13945574.99        1816775.       13945375.
      1815975.02     13944675.02
#Sta/Elev= 30
  4507.8 2070.83  4545.4 2070.03  4588.9 2058.76  4615.2 2050.94    4661 2041.26
  4713.6 2023.05  4748.5 2015.32  4781.4 2013.57  4794.3 2010.41  4835.4  2013.2
  4840.9 2011.31  4901.7 2009.44  4916.1 2006.62  4962.6 2006.59  4968.1 2004.14
    5000 2002.86  5000.5 2002.36  5027.9 2002.86    5050 2003.58  5085.2    2013
  5113.6 2015.37  5120.3 2018.75  5134.5 2020.33  5336.3 2022.46  5475.3 2020.59
  5531.7 2015.49  5559.7 2015.65  5857.7 2022.96  6000.8 2031.14  6063.2 2035.05
#Mann= 6 ,-1 , 0
  4507.8     .07       0  4588.9      .1       0    5000     .05       0
  5027.9      .1       0  5336.3     .07       0  6000.8      .1       0
#XS Ineff= 2 , 0
                          5300.9         2022.04
Permanent Ineff=
       F       F
Bank Sta=5000,5027.9
XS Rating Curve= 0 ,0
Exp/Cntr=0.3,0.1

Type RM Length L Ch R = 1 ,33566   ,555,555,555
BEGIN DESCRIPTION:
Bear Creek 2 58.0
END DESCRIPTION:
XS GIS Cut Line= 3
      1817425.02     13945475.04        1817225.       13945125.
      1815925.02     13944575.01
#Sta/Elev= 30
    4593  2075.2  4794.6 2070.19    4858 2067.18  4864.4 2064.84  4870.2 2058.26
  4880.3 2056.71    4886 2052.06  4901.9 2050.95  4907.6  2047.3  4923.5 2045.09
  4929.2 2038.34  4944.1 2032.31  4950.8 2026.63  4960.9 2023.48  4966.6 2007.25
  4973.1 2003.84  4996.2 2000.52  4996.8  1997.9  4997.3  1997.4  5024.7  1997.9
  5072.2 2008.01  5126.3 2010.18  5340.4 2019.97  5430.4 2020.07  5687.4 2015.17
  5745.4 2012.81  5897.4 2017.34  6010.7 2025.31  6284.4 2035.23  6407.7  2038.4
#Mann= 10 ,-1 , 0
    4593     .07       0  4794.6      .1       0  4944.1     .07       0
  4996.8     .05       0  5024.7     .07       0  5126.3      .1       0
  5340.4     .07       0  5430.4      .1       0  5687.4     .07       0
  6284.4      .1       0
#XS Ineff= 2 , 0
                         5383.12         2020.32
Permanent Ineff=
       F       F
Bank Sta=4996.8,5024.7
XS Rating Curve= 0 ,0
Exp/Cntr=0.3,0.1

Type RM Length L Ch R = 1 ,33011   ,527,527,527
BEGIN DESCRIPTION:
Bear Creek 2 57.0
END DESCRIPTION:
XS GIS Cut Line= 4
      1817575.02     13944825.02      1817355.48     13944618.52
        1817225.       13944625.      1815951.25     13944467.44
#Sta/Elev= 30
  4572.6 2052.14  4691.3 2050.25  4813.2 2045.64  4876.7 2039.93    4889 2037.53
  4906.7 2034.58  4924.5 2026.96  4944.6 2016.02  4954.6 2004.03  4970.7  1994.8
  4971.2  1994.3  4998.6  1994.8  5002.1 1997.55  5014.7 1999.63  5034.9 1999.42
  5085.2 2005.72  5115.5 2005.94  5196.1 2012.18  5377.5  2015.3  5417.8 2013.52
  5437.9 2009.61  5468.1 2012.09  5538.9 2012.78  5568.9 2011.15    5701  2013.4
    5782 2018.56  5863.1 2020.57  6020.1 2027.57  6182.2 2031.71  6288.1 2033.25
#Mann= 6 ,-1 , 0
  4572.6     .07       0  4691.3      .1       0    4889     .07       0
  4970.7     .05       0  4998.6     .07       0  6182.2      .1       0
#XS Ineff= 2 , 0
                         5355.04         2015.15
Permanent Ineff=
       F       F
Bank Sta=4970.7,4998.6
XS Rating Curve= 0 ,0
Exp/Cntr=0.3,0.1

Type RM Length L Ch R = 1 ,32484   ,576,576,576
BEGIN DESCRIPTION:
Bear Creek 2 56.0
END DESCRIPTION:
XS GIS Cut Line= 3
      1817475.01     13944325.01        1817125.       13944125.
      1816325.04     13943775.02
#Sta/Elev= 30
  4605.4 2036.53  4709.1 2027.92    4753 2027.72  4796.2 2020.14    4812 2019.74
  4817.8    2022  4840.1 2020.76  4876.8  2015.1  4898.4 2015.69  4914.2 2008.31
    4920 2010.64  4935.8 2002.05  4941.6  2004.4  4957.4 1997.17  4991.7 1994.81
  4992.2 1994.31  5019.7 1994.81  5040.9 1999.11  5098.6 1998.83  5145.4 2002.99
  5263.9 2005.42  5296.6 2005.15    5320  2008.3  5434.2 2009.28  5510.6 2006.05
  5554.3 2000.38  5608.9 2004.11  5674.7 2004.95  5797.1 2030.92  5881.7 2036.17
#Mann= 5 ,-1 , 0
  4605.4      .1       0  4840.1     .07       0  4991.7     .05       0
  5019.7     .07       0  5263.9      .1       0
#XS Ineff= 2 , 0
         4920.28 2010.46 5418.18         2009.36
Permanent Ineff=
       F       F
Bank Sta=4991.7,5019.7
XS Rating Curve= 0 ,0
Exp/Cntr=0.3,0.1

Type RM Length L Ch R = 1 ,31908   ,526,526,526
BEGIN DESCRIPTION:
Bear Creek 2 55.0
END DESCRIPTION:
XS GIS Cut Line= 3
      1817324.99       13943775.        1816925.       13943625.
      1816374.95       13943575.
#Sta/Elev= 30
  4572.4 2024.24  4743.3  2019.7  4828.7 2014.53  4838.5  2012.6  4874.1 2010.15
  4923.9 2000.27  4929.3 2000.97  4946.2 1997.23  4964.2  1995.3  4964.7  1994.8
  4992.2  1995.3  5019.7 1997.44    5110 1997.81  5150.2  2000.5  5200.2 1998.71
  5210.5 1999.57  5220.5 2002.84  5240.6 2004.33  5250.6 2003.61  5270.7 1997.21
  5280.7 1996.27  5310.9 2000.14  5330.9 1999.01  5371.1 2001.66  5381.2  2005.5
  5391.2 2011.97  5411.3 2019.43  5451.4 2030.03  5501.6 2037.51  5551.9 2039.95
#Mann= 4 ,-1 , 0
  4572.4     .07       0  4964.2     .05       0  4992.2     .07       0
  5200.2      .1       0
#XS Ineff= 2 , 0
                         5237.96         2004.27
Permanent Ineff=
       F       F
Bank Sta=4964.2,4992.2
XS Rating Curve= 0 ,0
Exp/Cntr=0.3,0.1

Type RM Length L Ch R = 1 ,31382   ,551,551,551
BEGIN DESCRIPTION:
Bear Creek 2 54.0
END DESCRIPTION:
XS GIS Cut Line= 3
      1817225.02     13943575.02        1816925.       13943175.
        1816975.     13942775.04
#Sta/Elev= 30
  4499.4 2016.46  4521.3 2015.18  4585.9 2014.22  4649.4 2012.07  4706.7 2007.71
  4730.1 2006.87  4771.3 2005.04  4806.7 2001.79  4835.9 2001.29  4856.7 1999.74
    4863 2000.39  4892.1 1999.96  4949.4 1994.32  4956.7 1991.82  4971.3 1989.88
  5029.7 1990.72  5034.7 1989.55  5035.2 1989.05    5065 1989.55  5090.1 2018.38
  5100.2 2024.47  5117.8 2030.87  5122.9  2029.5  5130.4 2032.73  5150.6 2037.79
  5180.8 2041.72  5314.8 2041.79    5320 2041.86  5326.7 2041.94  5402.5 2043.16
#Mann= 7 ,-1 , 0
  4499.4     .07       0  4730.1      .1       0  5034.7     .05       0
    5065      .1       0  5314.8     .07       0    5320      .1       0
  5326.7     .07       0
Bank Sta=5034.7,5065
XS Rating Curve= 0 ,0
Exp/Cntr=0.3,0.1

Type RM Length L Ch R = 1 ,30831   ,528,528,528
BEGIN DESCRIPTION:
Bear Creek 2 53.0
END DESCRIPTION:
XS GIS Cut Line= 3
        1817625.       13943475.        1817425.       13943125.
      1817124.98     13942824.98
#Sta/Elev= 30
  4597.4 2017.54  4670.1 2013.86  4707.5 2009.45    4745 2006.83  4750.7  2007.4
  4758.6 2005.67    4804 2001.17    4902 1996.42  4919.2 1995.88    4971 1993.32
  4977.5 1991.27  4992.6 1990.27  4997.6 1987.31    5004 1987.31  5013.6 1982.58
  5014.1 1982.08  5043.9 1982.58  5071.2 1985.21  5095.1 1994.52  5099.5 1996.37
  5113.6  2020.3  5127.8 2028.32  5141.9 2033.24  5170.2 2039.87  5198.5 2043.44
  5240.9  2044.5  5297.5 2044.81  5361.4 2043.13  5393.7 2042.84  5424.8 2042.85
#Mann= 8 ,-1 , 0
  4597.4     .07       0    4902      .1       0  4919.2     .07       0
  5013.6     .05       0  5043.9     .07       0  5095.1      .1       0
  5361.4     .07       0  5393.7      .1       0
Bank Sta=5013.6,5043.9
XS Rating Curve= 0 ,0
Exp/Cntr=0.3,0.1

Type RM Length L Ch R = 1 ,30303   ,582,582,582
BEGIN DESCRIPTION:
Bear Creek 2 52.0
END DESCRIPTION:
XS GIS Cut Line= 3
        1817925.     13943575.02        1817875.       13943175.
        1818025.     13942374.98
#Sta/Elev= 30
  4597.3 2024.72  4627.6 2024.26  4801.4 2015.45    4882 2004.95  4899.7 2001.44
  4929.9 1992.98  4957.6  1990.1  4990.4 1988.78  4995.4 1987.17  4995.9 1986.67
  5025.8 1987.17  5026.7 1988.69  5086.5 1989.11  5122.5 1988.81  5142.9  1990.1
  5189.5 2001.01  5214.1 2002.87  5242.1 2007.31  5247.2 2006.59  5294.6 2013.05
  5299.7 2012.67  5352.3 2020.86  5357.4 2020.35    5410 2027.36  5437.9 2033.02
  5498.2 2039.65  5580.4 2048.92  5724.5  2061.2  5788.1 2069.52  5814.4 2075.61
#Mann= 6 ,-1 , 0
  4597.3     .07       0  4995.4     .05       0  5025.8     .07       0
  5086.5      .1       0  5498.2     .07       0  5724.5      .1       0
Bank Sta=4995.4,5025.8
XS Rating Curve= 0 ,0
Exp/Cntr=0.3,0.1

Type RM Length L Ch R = 1 ,29721   ,565,565,565
BEGIN DESCRIPTION:
Bear Creek 2 51.0
END DESCRIPTION:
XS GIS Cut Line= 3
        1818425.       13943475.        1818425.       13943075.
        1818475.     13942624.97
#Sta/Elev= 30
  4599.6 2020.03  4639.6 2018.92  4749.6  2013.7  4819.6 2009.32  4849.6  2008.3
  4909.6 2000.84  4919.6 1998.83  4929.6 1995.34  4941.9 1989.43  4949.6 1984.84
  4959.6    1982  4964.4 1978.81  4964.9 1978.31  4994.3 1978.31  4994.8 1978.81
  4997.1 1981.05  5002.1 1981.05  5019.7  1984.1  5039.9 1985.85  5160.6 1992.24
  5210.9 2001.41  5241.1 2006.11  5251.1  2008.6  5281.3 2013.38  5291.4 2016.21
  5301.5 2018.21  5311.5 2019.46  5402.1 2036.69  5422.2 2039.43  5452.4 2042.08
#Mann= 4 ,-1 , 0
  4599.6     .07       0  4941.9      .1       0  4964.4     .05       0
  4994.8      .1       0
Bank Sta=4964.4,4994.8
XS Rating Curve= 0 ,0
Exp/Cntr=0.3,0.1

Type RM Length L Ch R = 1 ,29156   ,527,527,527
BEGIN DESCRIPTION:
Bear Creek 2 50.0
END DESCRIPTION:
XS GIS Cut Line= 3
      1818690.03      13943488.8        1818925.       13942975.
      1819224.97     13942675.03
#Sta/Elev= 30
  4438.8 2017.63    4498  2016.3  4558.7 2013.59  4574.9 2013.79  4604.7 2011.19
  4656.3 2009.81  4776.9 2002.96  4799.9 2001.14  4805.8 1999.45  4838.8 1994.75
  4845.2 1992.89  4860.8 1991.78  4868.9 1986.97  4891.9 1982.07  4937.8 1982.64
  4959.8 1981.37  4966.5 1980.54  4966.6 1979.79  4967.1 1979.29    4997 1979.79
    5001 1981.34  5017.9 1982.63  5074.5 1983.34  5131.1 1987.98  5187.6 1999.11
  5244.2 2012.64  5258.3 2014.64  5286.6 2021.43  5385.6 2036.53    5428 2041.75
#Mann= 4 ,-1 , 0
  4438.8     .07       0  4845.2      .1       0  4966.6     .05       0
    4997      .1       0
Bank Sta=4966.6,4997
XS Rating Curve= 0 ,0
Exp/Cntr=0.3,0.1

Type RM Length L Ch R = 1 ,28629   ,523,523,523
BEGIN DESCRIPTION:
Bear Creek 2 49.0
END DESCRIPTION:
XS GIS Cut Line= 3
      1818802.75     13943489.38        1819375.       13943025.
      1819475.01     13942624.98
#Sta/Elev= 30
  4258.8 2015.52  4349.2 2012.55  4398.8 2009.31  4611.4 2002.43  4689.7 1997.48
    4712  1997.3  4753.6 1993.89  4796.8 1993.52  4811.1 1992.18  4817.6 1990.05
  4825.5 1989.39    4832 1986.16  4846.3 1983.98  4859.5 1984.09  4931.4 1980.58
  4967.8 1980.92  4998.3 1978.92  5003.7 1977.53  5004.2 1977.03  5034.2 1977.53
    5037 1979.16  5060.2 1981.74  5078.2 1999.99  5096.3 2011.06  5119.5 2023.01
  5160.7 2034.72    5220 2043.14  5261.2  2044.1  5315.3 2048.55  5408.1 2053.18
#Mann= 4 ,-1 , 0
  4258.8     .07       0  4859.5      .1       0  5003.7     .05       0
  5034.2      .1       0
Bank Sta=5003.7,5034.2
XS Rating Curve= 0 ,0
Exp/Cntr=0.3,0.1

Type RM Length L Ch R = 1 ,28106   ,523,523,523
BEGIN DESCRIPTION:
Bear Creek 2 48.0
END DESCRIPTION:
XS GIS Cut Line= 3
      1819574.99     13943625.02        1819825.       13943225.
        1819825.     13942825.02
#Sta/Elev= 30
  4523.5  2008.6  4594.9 2004.52  4625.5  2000.7  4698.6 1996.64  4725.8 1994.36
  4777.7  1992.4  4783.5    1993  4835.4 1990.57  4850.8 1988.59  4877.9 1982.19
  4899.2 1981.52  4914.4  1980.1  4945.1 1979.54  4972.2 1977.13  4987.6 1977.08
  4992.3 1975.31  4997.7 1975.31  4999.9 1973.76  5000.4 1973.26  5030.5 1973.76
  5035.2 1976.02  5065.2 1979.47  5075.2 1984.29  5085.2 1995.57  5095.2 2000.46
  5145.2 2018.15  5175.2 2024.92  5205.2 2029.93  5255.2 2035.97  5395.2 2043.43
#Mann= 4 ,-1 , 0
  4523.5     .07       0  4899.2      .1       0  4999.9     .05       0
  5030.5      .1       0
Bank Sta=4999.9,5030.5
XS Rating Curve= 0 ,0
Exp/Cntr=0.3,0.1

Type RM Length L Ch R = 1 ,27583   ,585,585,585
BEGIN DESCRIPTION:
Bear Creek 2 47.0
END DESCRIPTION:
XS GIS Cut Line= 3
      1819974.99     13944025.02        1820275.       13943425.
      1820625.04     13943224.98
#Sta/Elev= 30
  4333.1  2013.2    4434 2007.64  4475.7 2005.59  4539.3 1999.69  4580.3 1997.39
  4647.5 1993.19  4766.4  1987.5  4809.6 1979.82  4847.4 1977.89  4861.4 1978.44
  4869.8 1976.68  4950.8 1975.35  4966.2 1973.45  4966.7 1972.95  4996.9 1973.45
  5001.1 1975.11  5011.9 1975.99    5027 1979.93  5033.5 1983.19  5039.2 1989.48
    5055 1994.68  5076.6 1999.59  5107.6 2004.79  5119.8 2008.79  5135.7 2010.55
  5178.9 2019.14  5253.7 2030.63  5281.1 2033.71  5312.8 2036.23  5407.1 2038.43
#Mann= 8 ,-1 , 0
  4333.1     .07       0    4434      .1       0  4539.3     .07       0
  4580.3      .1       0  4647.5     .07       0  4809.6      .1       0
  4966.2     .05       0  4996.9      .1       0
Bank Sta=4966.2,4996.9
XS Rating Curve= 0 ,0
Exp/Cntr=0.3,0.1

Type RM Length L Ch R = 1 ,26998   ,747,747,747
BEGIN DESCRIPTION:
Bear Creek 2 46.0
END DESCRIPTION:
XS GIS Cut Line= 3
      1820475.02     13944174.96        1820675.       13943825.
        1820675.     13943324.97
#Sta/Elev= 30
  4596.9 2006.22  4624.6 2004.04  4663.8 2000.24  4771.8 1984.39  4787.6 1983.44
  4815.7 1979.99  4838.7 1980.41  4868.2 1975.83  4942.4 1972.81  4954.6 1971.92
  4955.1 1970.93  4955.6 1970.43  4985.8 1970.93  4986.3  1971.9  4997.1 1973.42
    5030 1974.07    5050 1973.52    5080 1975.07    5100 1977.11    5120 1980.74
    5130  1984.1    5160 1990.91    5180 1993.15    5200 1993.89    5270  2000.6
    5340 2011.22    5380 2018.69    5430 2025.42    5480 2033.71    5500 2035.03
#Mann= 4 ,-1 , 0
  4596.9     .07       0  4624.6      .1       0  4955.1     .05       0
  4985.8      .1       0
Bank Sta=4955.1,4985.8
XS Rating Curve= 0 ,0
Exp/Cntr=0.3,0.1

Type RM Length L Ch R = 1 ,26251   ,400,400,400
BEGIN DESCRIPTION:
Bear Creek 2 45.1
END DESCRIPTION:
XS GIS Cut Line= 3
      1821312.32     13944642.64      1821218.11     13944087.26
      1821059.02     13943369.29
#Sta/Elev= 30
  4575.9 2030.59  4594.3 2027.56  4715.5 2014.91  4756.1 2012.15  4890.9 1999.33
  4918.4  1993.3  4928.5 1980.82  4946.1 1968.01  4958.9 1967.31  4973.7 1963.05
  4974.2 1962.55    5005 1963.05  5006.5  1964.4  5011.5 1964.01  5019.8 1966.23
  5071.9 1968.62  5090.8 1971.11  5111.1 1971.87  5121.2 1973.49  5127.1 1975.77
  5132.2 1975.34  5137.8 1977.53    5177 1978.42    5220 1981.79  5269.4 1983.95
  5366.9 1991.69  5612.7 2000.83  5766.3 2011.95  5786.8 2014.99  5874.6 2022.27
#Mann= 4 ,-1 , 0
  4575.9      .1       0  4973.7     .05       0    5005      .1       0
    5220     .07       0
Bank Sta=4973.7,5005
XS Rating Curve= 0 ,0
Exp/Cntr=0.3,0.1

Type RM Length L Ch R = 1 ,25851   ,542,542,542
BEGIN DESCRIPTION:
Bear Creek 2 45.0
END DESCRIPTION:
XS GIS Cut Line= 3
        1821825.       13944625.        1821625.       13944275.
        1821625.     13943875.01
#Sta/Elev= 30
  4596.9 2037.32    4648 2031.65  4654.5 2030.08  4700.6 2024.35  4712.8 2021.92
  4744.5 2018.58  4771.8 2013.43  4825.1 2008.21  4905.7 1996.81  4933.1 1990.62
  4948.9 1982.82  4954.7 1982.68  4964.7 1974.35  4970.5 1973.13    4977 1962.29
  4986.3 1961.49  4992.1 1961.94  4994.4 1959.05  4994.9 1958.55  5025.7 1959.05
    5030 1962.36    5040 1964.24    5050 1963.85    5090 1968.73    5160 1972.65
    5210 1979.32    5280 1982.34    5300  1985.6    5350 1989.98    5400 1991.88
#Mann= 3 ,-1 , 0
  4596.9      .1       0  4994.4     .05       0  5025.7      .1       0
Bank Sta=4994.4,5025.7
XS Rating Curve= 0 ,0
Exp/Cntr=0.3,0.1

Type RM Length L Ch R = 1 ,25309   ,555,555,555
BEGIN DESCRIPTION:
Bear Creek 2 44.0
END DESCRIPTION:
XS GIS Cut Line= 3
      1822024.99     13944625.03        1822125.       13944225.
        1822125.     13943825.04
#Sta/Elev= 30
  4593.3 2043.33  4616.5 2043.55  4634.6 2042.45  4665.5 2037.54  4686.1 2035.88
  4693.8 2033.94    4851 2018.36  4881.9 2013.29  4892.3 2010.56    4900 2006.44
  4905.1 2006.41  4923.2  1998.9  4933.5 1991.41  4941.2  1984.4  4946.4 1984.81
  4964.4 1965.92  4966.7 1958.66  4967.2 1958.16  4998.1 1958.66  5003.1 1959.74
  5055.6 1963.02  5115.6 1964.65  5155.6 1968.38  5175.6 1971.83  5195.6 1973.88
  5215.6 1978.17  5245.6 1979.48  5295.6 1985.14  5355.6 1990.09  5405.6 1991.14
#Mann= 3 ,-1 , 0
  4593.3      .1       0  4966.7     .05       0  4998.1      .1       0
Bank Sta=4966.7,4998.1
XS Rating Curve= 0 ,0
Exp/Cntr=0.3,0.1

Type RM Length L Ch R = 1 ,24754   ,505,505,505
BEGIN DESCRIPTION:
Bear Creek 2 43.0
END DESCRIPTION:
XS GIS Cut Line= 3
      1822974.97     13944274.99        1822625.       13944075.
        1822425.       13943725.
#Sta/Elev= 30
  4591.3 2033.72    4664 2030.68  4766.2 2023.18  4819.5 2016.45  4856.2 2006.65
  4862.7 2004.03  4868.4 2000.13  4878.5 1997.09  4890.7 1988.36  4900.1 1984.81
  4905.8 1980.39  4921.7 1972.89  4927.4  1967.5    4949 1960.28  4970.7 1958.99
  4971.2 1958.49  5002.2 1958.99  5002.3 1960.05  5017.4 1960.94  5029.7 1959.82
  5067.1 1959.52  5126.1  1962.5    5142 1966.52  5178.7 1971.29  5213.2 1977.89
  5259.3 1981.07  5281.6 1983.74  5346.4  1987.7  5374.5  1991.2  5397.5 1991.46
#Mann= 3 ,-1 , 0
  4591.3      .1       0  4970.7     .05       0  5002.2      .1       0
Bank Sta=4970.7,5002.2
XS Rating Curve= 0 ,0
Exp/Cntr=0.3,0.1

Type RM Length L Ch R = 1 ,24249   ,587,587,587
BEGIN DESCRIPTION:
Bear Creek 2 42.0
END DESCRIPTION:
XS GIS Cut Line= 3
        1823025.     13944225.02        1823025.       13943825.
      1822675.03     13943575.02
#Sta/Elev= 30
  4594.7 2033.18  4624.7 2031.95  4734.7 2023.93  4754.7 2023.24  4764.7 2021.59
  4814.7 2017.89  4864.7 2011.71  4874.7 2009.68  4894.7 2001.76  4944.7 1977.63
  4954.7 1964.04  4964.7 1959.58  4974.7 1957.88  4997.8 1956.06  5001.1 1953.51
  5001.6 1953.01  5032.6 1953.51  5043.9 1955.85  5052.5 1955.43  5073.4 1956.56
    5109 1960.18  5117.6 1959.72  5166.8 1968.14  5252.8  1972.3  5289.7 1975.73
  5301.9 1978.74  5310.5 1979.41  5360.9 1980.76    5388 1984.02  5424.8 1985.66
#Mann= 3 ,-1 , 0
  4594.7      .1       0  5001.1     .05       0  5032.6      .1       0
Bank Sta=5001.1,5032.6
XS Rating Curve= 0 ,0
Exp/Cntr=0.3,0.1

Type RM Length L Ch R = 1 ,23662   ,531,531,531
BEGIN DESCRIPTION:
Bear Creek 2 41.0
END DESCRIPTION:
XS GIS Cut Line= 3
        1823725.       13943575.        1823375.       13943375.
      1822975.01     13943125.01
#Sta/Elev= 30
  4601.5 2045.71  4624.5 2044.12    4631 2042.07    4690 2034.51  4727.5 2028.28
  4785.8 2023.06    4798 2020.22  4820.3 2018.22  4866.4 2010.67  4894.5 2000.99
  4931.9 1977.63  4937.7 1973.04    4947  1960.3  4953.5 1956.39  4974.9 1949.89
  4975.4 1949.39    5007 1949.89  5012.3  1953.6  5018.2 1954.22    5040 1954.58
  5091.3 1959.49    5099 1958.13  5121.9 1959.13  5206.9 1967.52    5280 1971.57
  5310.6 1974.37  5331.9 1978.89    5382  1979.5  5426.2  1984.8  5476.3 1986.67
#Mann= 3 ,-1 , 0
  4601.5      .1       0  4974.9     .05       0    5007      .1       0
Bank Sta=4974.9,5007
XS Rating Curve= 0 ,0
Exp/Cntr=0.3,0.1

Type RM Length L Ch R = 1 ,23131   ,505,505,505
BEGIN DESCRIPTION:
Bear Creek 2 40.0
END DESCRIPTION:
XS GIS Cut Line= 3
        1823825.       13943275.        1823625.       13942925.
      1823375.01     13942575.02
#Sta/Elev= 30
  4602.9 2030.77    4654 2024.15  4750.5 2007.55  4799.4 2001.44  4852.7 1990.93
    4880 1980.47  4890.1 1978.71  4895.9 1974.78  4911.7  1969.6  4917.5 1964.36
  4933.3 1958.23  4939.1  1954.5  4954.9 1954.48  4960.7 1950.18  4966.8 1947.68
  4967.4 1947.18  4999.1 1947.68  5003.1 1951.02  5034.3 1953.13  5141.2 1955.66
  5149.8 1956.65  5170.7 1963.53  5191.6 1968.29  5235.8 1971.46    5242 1973.54
  5277.6 1978.87  5345.1 1983.28  5372.2 1985.21  5399.3 1989.48  5436.1 1991.32
#Mann= 4 ,-1 , 0
  4602.9      .1       0  4966.8     .05       0  4999.1      .1       0
  5345.1     .07       0
Bank Sta=4966.8,4999.1
XS Rating Curve= 0 ,0
Exp/Cntr=0.3,0.1

Type RM Length L Ch R = 1 ,22626   ,639,639,639
BEGIN DESCRIPTION:
Bear Creek 2 39.0
END DESCRIPTION:
XS GIS Cut Line= 3
      1824274.98     13942774.99      1823944.96     13942558.22
      1823624.96     13942274.97
#Sta/Elev= 30
  4567.7 2038.36  4647.5  2030.6  4683.7 2025.04  4719.9  2017.9    4807 1997.37
  4819.2 1993.23  4828.4 1992.13  4842.9 1988.19  4885.6 1975.61  4900.7 1969.65
  4927.7 1956.88  4950.5    1952  4965.9 1952.68  4970.1 1949.19  4970.6 1948.69
  5002.4 1949.19  5049.8 1950.48  5120.9 1949.52  5127.6 1950.37  5135.2 1953.58
  5141.8 1954.92  5149.4 1957.75  5162.8 1965.16    5177 1969.62  5198.7 1972.45
    5213 1975.81  5227.2 1977.67  5283.2 1980.83  5333.4  1986.4  5389.9 1989.61
#Mann= 3 ,-1 , 0
  4567.7      .1       0  4970.1     .05       0  5002.4      .1       0
Bank Sta=4970.1,5002.4
XS Rating Curve= 0 ,0
Exp/Cntr=0.3,0.1

Type RM Length L Ch R = 1 ,21987   ,585,585,585
BEGIN DESCRIPTION:
Bear Creek 2 38.0
END DESCRIPTION:
XS GIS Cut Line= 3
      1824375.01     13942675.02        1824175.       13942025.
        1823975.     13941675.01
#Sta/Elev= 30
  4319.9 2029.14  4351.3 2025.54  4401.7 2016.64  4445.5  2011.6  4487.3 2003.65
    4575 1993.32  4633.8  1984.7  4654.7 1979.91  4678.9 1977.15  4717.5 1967.78
  4738.4 1965.33  4759.4 1958.09  4782.2 1953.83  4814.9 1950.46  4874.4 1950.79
  4937.2 1948.55  4978.4 1943.85  4981.2 1942.13  4981.7 1941.63  5013.6 1942.13
  5013.7 1944.43  5029.5 1946.21  5045.3 1950.73  5057.6  1958.6  5066.9 1967.11
  5072.7 1970.02  5094.3 1975.18  5147.6 1978.89  5255.5 1989.65  5403.1 1996.44
#Mann= 3 ,-1 , 0
  4319.9      .1       0  4981.2     .05       0  5013.6      .1       0
Bank Sta=4981.2,5013.6
XS Rating Curve= 0 ,0
Exp/Cntr=0.3,0.1

Type RM Length L Ch R = 1 ,21402   ,227,227,227
BEGIN DESCRIPTION:
Bear Creek 2 37.0
END DESCRIPTION:
XS GIS Cut Line= 3
      1824674.99     13942024.97        1824575.       13941625.
      1824174.99       13941525.
#Sta/Elev= 30
  4588.2 1986.21  4722.2 1977.18  4771.1 1972.18  4776.3 1970.14  4804.6 1967.73
  4825.3 1961.09  4845.9 1958.11  4866.5  1953.2  4894.8 1952.55    4918 1950.28
  4941.2 1946.45  4969.6 1944.72  4997.9 1938.39  5031.4 1938.08  5041.7 1938.81
  5048.7 1937.96  5049.3 1937.46  5081.1 1937.96  5093.3 1939.17    5101 1942.01
  5124.2 1945.74  5155.1 1954.75  5188.6 1962.83  5196.3 1966.75  5224.7  1969.7
  5229.8 1969.57  5258.2 1974.87  5340.6 1982.78  5389.6 1989.36  5412.8 1990.42
#Mann= 3 ,-1 , 0
  4588.2      .1       0  5048.7     .05       0  5081.1      .1       0
Bank Sta=5048.7,5081.1
XS Rating Curve= 0 ,0
Exp/Cntr=0.3,0.1

Type RM Length L Ch R = 1 ,21175   ,838,838,838
BEGIN DESCRIPTION:
Bear Creek 2 36.1
END DESCRIPTION:
XS GIS Cut Line= 3
      1825304.68     13941648.18      1824757.86     13941437.27
      1824224.17     13941358.19
#Sta/Elev= 30
  4287.9 1980.36  4351.9 1977.83  4476.2 1968.29  4536.2 1965.64  4576.9 1962.52
    4670 1958.27  4779.1 1955.95  4839.1 1952.31  4844.9 1950.25  4872.8  1945.2
    4878  1945.2  4897.1 1940.45  4947.6 1937.06  4967.9 1934.12  4972.3 1932.42
  4973.3 1931.92  5012.6 1932.42  5018.4 1938.64  5038.6  1939.4    5062 1945.68
  5089.2 1949.78  5159.9 1957.86  5190.3  1963.5  5195.9 1966.24    5201 1965.91
  5240.8 1970.36  5271.1 1975.76  5281.2 1975.85  5382.3 1988.03  5413.5 1990.56
#Mann= 3 ,-1 , 0
  4287.9      .1       0  4972.3     .05       0  5012.6      .1       0
Bank Sta=4972.3,5012.6
XS Rating Curve= 0 ,0
Exp/Cntr=0.3,0.1
