--- Bee Caves Creek.prj (project) ---

Proj Title=Bee Caves Creek Base Level Engineering
Current Plan=p01
Default Exp/Contr=0.3,0.1
English Units
Geom File=g01
Flow File=f01
Plan File=p01
BEGIN DESCRIPTION:
Bee Caves Creek
END DESCRIPTION:

--- Bee Caves Creek.p01 (plan) ---

Plan Title=Multiple Run
Short Identifier=Multiple
Geom File=g01
Flow File=f01
Subcritical Flow
K Sum by GR= 0
Std Step Tol= 0.01
Critical Tol= 0.01
Num of Std Step Trials= 20
Max Error Tol= 0.3
Flow Tol Ratio= 0.001
Split Flow NTrial= 30
Split Flow Tol= 0.02
Split Flow Ratio= 0.02
Log Output Level= 0
Friction Slope Method= 1
Unsteady Friction Slope Method= 2
Unsteady Bridges Friction Slope Method= 1
Parabolic Critical Depth
Global Vel Dist=  1 , 1 , 1
Global Log Level= 0
CheckData=True
Encroach Param= -1, 0, 0, 0
BEGIN DESCRIPTION:
Multiple Run
END DESCRIPTION:

--- Bee Caves Creek.f01 (steady flow) ---

Flow Title=Multiple
Number of Profiles=7
Profile Names=10-year,25-year,50-year,1pct_min,100-year,1pct_plu,500-year
River Rch & RM= Bee Caves Creek,Reach-1,29493
     287     452     597     384     765    1527    1237
River Rch & RM= Bee Caves Creek,Reach-1,27636
    1318    2296    3242    2212    4413    8805    8087
River Rch & RM= Bee Caves Creek,Reach-1,21193
    1954    3468    4960    3420    6824   13615   12787
River Rch & RM= Bee Caves Creek,Reach-1,17480
    2351    4205    6044    4185    8350   16660   15779
River Rch & RM= Bee Caves Creek,Reach-1,13758
    3443    6246    9063    6325   12620   25180   24238
River Rch & RM= Bee Caves Creek,Reach-1,5545
    3467    6282    9106    6348   12666   25271   24272
Boundary for River Rch & Prof#=Bee Caves Creek,Reach-1,1
Up Type=0
Dn Type=3
Dn Slope=0.005
Boundary for River Rch & Prof#=Bee Caves Creek,Reach-1,2
Up Type=0
Dn Type=3
Dn Slope=0.005
Boundary for River Rch & Prof#=Bee Caves Creek,Reach-1,3
Up Type=0
Dn Type=3
Dn Slope=0.005
Boundary for River Rch & Prof#=Bee Caves Creek,Reach-1,4
Up Type=0
Dn Type=3
Dn Slope=0.005
Boundary for River Rch & Prof#=Bee Caves Creek,Reach-1,5
Up Type=0
Dn Type=3
Dn Slope=0.005
Boundary for River Rch & Prof#=Bee Caves Creek,Reach-1,6
Up Type=0
Dn Type=3
Dn Slope=0.005
Boundary for River Rch & Prof#=Bee Caves Creek,Reach-1,7
Up Type=0
Dn Type=3
Dn Slope=0.005

--- Bee Caves Creek.g01 (geometry) ---

Geom Title=Existing Conditions

River Reach=Bee Caves Creek,Reach-1
Reach XY= 30
      1813625.00     13914175.00      1814077.74     13914180.34
      1814368.83     13914567.14      1815664.35     13915265.00
      1815925.30     13916095.18      1815776.20     13916764.50
      1816230.83     13918177.30      1817091.65     13919391.67
      1817948.71     13919948.18      1818138.54     13920538.38
      1818921.85     13921233.32      1819024.49     13921609.78
      1818724.57     13923109.82      1818885.61     13924035.06
      1820664.50     13924026.20      1821271.24     13924426.56
      1821421.47     13924973.53      1820630.54     13925722.58
      1820524.96     13926505.02      1821722.94     13927380.85
      1821571.25     13928323.45      1820924.76     13929100.08
      1821338.40     13930188.30      1822272.84     13930730.97
      1821882.56     13932175.00      1821980.46     13932877.45
      1822209.58     13933074.97      1823309.78     13932725.49
      1823950.00     13933125.42      1824225.00     13932875.00

Type RM Length L Ch R = 1,29493,464,464,464
BEGIN DESCRIPTION:
Bee Caves Creek 64.0
END DESCRIPTION:
XS GIS Cut Line= 3
      1813475.02     13914424.98      1813775.00     13914175.00
      1813825.00     13913574.97
#Sta/Elev= 30
  4609.5 2219.62  4631.0 2217.23  4637.5 2217.80  4645.3 2216.11  4680.4 2214.81
  4694.7 2213.10  4729.9 2211.65  4779.3 2208.40  4908.2 2204.21  4921.9 2204.63
  4929.0 2203.59  4972.0 2201.84  5050.2 2199.83  5080.3 2200.31  5130.4 2199.73
  5158.5 2198.18  5158.8 2197.68  5162.5 2198.18  5183.1 2198.38  5220.8 2201.53
  5230.8 2201.26  5311.1 2203.93  5371.3 2208.17  5391.3 2208.81  5418.9 2212.27
  5437.4 2213.49  5535.9 2223.45  5572.0 2225.94  5582.0 2225.72  5602.1 2226.90
#Mann=5,-1,0
  4609.5     0.1       0  5158.5    0.05       0  5162.5     0.1       0
  5437.4    0.07       0  5535.9     0.1       0
Bank Sta=5158.5,5162.5
Exp/Cntr=0.3,0.1

Type RM Length L Ch R = 1,29029,448,448,448
BEGIN DESCRIPTION:
Bee Caves Creek 63.0
END DESCRIPTION:
XS GIS Cut Line= 3
      1813825.02     13914624.98      1814125.00     13914325.00
      1814425.00     13914025.00
#Sta/Elev= 30
  4571.4 2214.01  4574.9 2214.01  4599.7 2210.16  4627.9 2207.14  4656.2 2205.14
  4698.6 2200.91  4726.9 2199.92  4741.1 2198.52  4769.4 2197.25  4811.8 2193.98
  4825.9 2193.64  4854.2 2191.05  4896.6 2189.10  4958.7 2187.68  4990.1 2186.98
  4990.3 2186.48  4993.8 2186.48  4994.1 2186.98  5038.1 2187.63  5052.2 2187.22
  5080.5 2188.22  5094.6 2189.52  5122.9 2190.81  5173.0 2192.03  5207.8 2193.55
  5236.0 2193.68  5292.6 2196.17  5335.0 2199.76  5384.5 2202.54  5419.9 2206.63
#Mann=5,-1,0
  4571.4     0.1       0  4958.7   0.035       0  4990.1   0.035       0
  4994.1   0.035       0  5173.0     0.1       0
Bank Sta=4990.1,4994.1
Exp/Cntr=0.3,0.1

Type RM Length L Ch R = 1,28581,476,476,476
BEGIN DESCRIPTION:
Bee Caves Creek 62.0
END DESCRIPTION:
XS GIS Cut Line= 3
      1814175.00     13914775.00      1814475.00     13914575.00
      1814774.98     13914275.02
#Sta/Elev= 30
  4644.4 2197.23  4672.9 2196.32  4694.0 2193.27  4760.1 2189.19  4796.1 2188.70
  4817.2 2186.12  4853.2 2184.67  4874.3 2183.15  4919.3 2181.47  4932.8 2181.73
  4968.9 2180.72  5000.0 2177.37  5000.2 2176.87  5003.7 2176.87  5004.0 2177.37
  5012.1 2177.66  5061.5 2180.44  5075.7 2180.31  5089.8 2181.30  5118.1 2182.03
  5160.5 2184.50  5217.1 2186.81  5233.2 2188.09  5245.4 2188.55  5273.7 2191.70
  5301.9 2193.15  5314.1 2194.52  5330.2 2194.84  5400.9 2200.97  5429.2 2202.58
#Mann=6,-1,0
  4644.4    0.07       0  5000.0    0.05       0  5004.0    0.07       0
  5012.1   0.035       0  5233.2    0.07       0  5314.1     0.1       0
Bank Sta=5000,5004
Exp/Cntr=0.3,0.1

Type RM Length L Ch R = 1,28105,469,469,469
BEGIN DESCRIPTION:
Bee Caves Creek 61.0
END DESCRIPTION:
XS GIS Cut Line= 3
      1814574.98     13915075.02      1814875.00     13914775.00
      1814974.99     13914475.02
#Sta/Elev= 30
  4575.4 2190.94  4646.1 2187.24  4688.6 2182.88  4731.0 2180.93  4759.3 2178.93
  4822.9 2176.12  4886.6 2174.83  4929.0 2172.53  4957.3 2172.26  4985.5 2171.00
  4996.2 2168.79  5008.2 2168.21  5008.5 2167.71  5012.0 2167.71  5012.2 2168.21
  5020.8 2169.49  5031.3 2171.91  5052.4 2173.69  5084.0 2175.14  5094.6 2175.00
  5147.3 2177.00  5168.3 2179.19  5178.9 2179.96  5189.4 2179.89  5210.1 2181.78
  5242.1 2182.99  5263.2 2184.67  5273.8 2186.18  5294.8 2188.04  5315.9 2188.78
#Mann=4,-1,0
  4575.4   0.035       0  5008.2   0.035       0  5012.2   0.035       0
  5210.1    0.07       0
Bank Sta=5008.2,5012.2
Exp/Cntr=0.3,0.1

Type RM Length L Ch R = 1,27636,446,446,446
BEGIN DESCRIPTION:
Bee Caves Creek 60.0
END DESCRIPTION:
XS GIS Cut Line= 3
      1814924.97     13915375.03      1815225.00     13915075.00
      1815225.00     13914775.01
#Sta/Elev= 30
  4575.9 2187.74  4646.7 2181.05  4660.8 2180.58  4717.4 2176.12  4759.8 2174.21
  4802.2 2173.21  4816.4 2172.47  4844.6 2169.55  4901.2 2165.70  4943.6 2163.69
  4957.8 2163.53  4996.7 2161.35  5008.2 2161.34  5008.5 2160.84  5012.0 2160.84
  5012.2 2161.34  5020.2 2162.87  5060.2 2163.00  5080.2 2161.99  5090.2 2162.77
  5100.2 2165.19  5130.2 2167.69  5140.2 2167.28  5170.2 2168.38  5180.2 2168.20
  5220.2 2169.24  5230.2 2169.89  5250.2 2170.16  5290.2 2172.22  5300.2 2172.24
#Mann=3,-1,0
  4575.9    0.07       0  5008.2    0.05       0  5012.2    0.07       0
Bank Sta=5008.2,5012.2
Exp/Cntr=0.3,0.1

Type RM Length L Ch R = 1,27190,471,471,471
BEGIN DESCRIPTION:
Bee Caves Creek 59.0
END DESCRIPTION:
XS GIS Cut Line= 3
      1815330.65     13915402.71      1815625.00     13915225.00
      1815898.31     13914944.46
#Sta/Elev= 30
  4661.6 2168.63  4706.6 2166.50  4743.4 2163.51  4795.2 2161.44  4844.4 2158.31
  4902.6 2156.58  4912.0 2155.61  4918.1 2153.99  4923.9 2154.04  4955.0 2150.02
  4970.4 2147.36  4982.2 2144.29  4989.8 2143.51  4990.1 2143.01  4993.6 2143.01
  4993.8 2143.51  4997.7 2144.88  5002.5 2147.72  5008.9 2147.72  5012.5 2151.02
  5033.6 2154.32  5040.8 2156.38  5061.9 2159.59  5111.5 2165.23  5139.8 2166.50
  5160.9 2168.43  5224.7 2172.28  5302.4 2174.80  5323.7 2174.77  5397.1 2177.71
#Mann=3,-1,0
  4661.6    0.07       0  4989.8    0.05       0  4993.8    0.07       0
Bank Sta=4989.8,4993.8
Exp/Cntr=0.3,0.1

Type RM Length L Ch R = 1,26719,434,434,434
BEGIN DESCRIPTION:
Bee Caves Creek 58.0
END DESCRIPTION:
XS GIS Cut Line= 3
      1815245.82     13915707.41      1815725.00     13915625.00
      1816255.40     13915615.59
#Sta/Elev= 30
  4519.1 2175.16  4569.0 2172.22  4678.2 2168.27  4751.6 2162.63  4803.1 2160.87
  4832.8 2158.14  4858.0 2156.77  4917.9 2150.78  4924.1 2149.37  4934.3 2148.28
  4972.8 2137.24  4977.9 2137.99  4983.0 2135.22  4983.3 2134.72  4986.8 2134.72
  4987.0 2135.22  4995.2 2137.59  5002.8 2138.79  5025.3 2140.30  5065.3 2145.63
  5095.3 2148.21  5165.3 2152.34  5205.3 2153.50  5225.3 2155.95  5255.4 2156.86
  5283.7 2159.49  5315.4 2161.30  5345.4 2164.97  5385.4 2166.44  5535.8 2176.41
#Mann=3,-1,0
  4519.1    0.07       0  4983.0    0.05       0  4987.0    0.07       0
Bank Sta=4983,4987
Exp/Cntr=0.3,0.1

Type RM Length L Ch R = 1,26285,461,461,461
BEGIN DESCRIPTION:
Bee Caves Creek 57.0
END DESCRIPTION:
XS GIS Cut Line= 3
      1815574.97     13915975.00      1815875.00     13915975.00
      1816264.69     13915841.02
#Sta/Elev= 30
  4704.7 2158.71  4764.7 2154.65  4774.7 2152.67  4794.7 2150.76  4864.7 2145.62
  4894.7 2141.33  4904.7 2141.12  4934.7 2137.93  4954.7 2133.29  4992.7 2132.06
  4993.0 2131.56  4996.7 2132.06  5007.4 2132.11  5020.3 2134.37  5046.3 2141.25
  5051.6 2141.38  5057.6 2145.06  5077.5 2149.66  5082.8 2149.74  5106.9 2153.29
  5140.0 2157.40  5176.5 2160.04  5226.8 2165.21  5233.7 2166.94  5239.0 2166.56
  5265.0 2170.22  5311.4 2173.17  5364.3 2178.34  5389.9 2179.65  5416.8 2182.92
#Mann=4,-1,0
  4704.7    0.07       0  4992.7    0.05       0  4996.7    0.07       0
  5106.9     0.1       0
Bank Sta=4992.7,4996.7
Exp/Cntr=0.3,0.1

Type RM Length L Ch R = 1,25824,407,407,407
BEGIN DESCRIPTION:
Bee Caves Creek 56.0
END DESCRIPTION:
XS GIS Cut Line= 3
      1815675.03     13916375.00      1815775.00     13916375.00
      1816075.01     13916275.00
#Sta/Elev= 30
  4894.3 2147.31  4896.8 2147.31  4924.3 2140.48  4934.3 2138.32  4954.3 2134.26
  4964.3 2132.76  4984.3 2128.61  4991.8 2126.31  4996.9 2126.31  5004.8 2125.26
  5023.9 2124.95  5024.1 2124.45  5027.6 2124.45  5027.9 2124.95  5057.5 2127.51
  5068.1 2129.55  5078.6 2130.15  5089.1 2131.43  5110.2 2132.64  5131.3 2136.33
  5152.4 2139.30  5162.9 2141.15  5173.5 2143.82  5226.2 2150.23  5236.7 2152.20
  5257.8 2154.42  5268.3 2155.95  5300.0 2159.05  5307.9 2160.28  5310.5 2160.28
#Mann=3,-1,0
  4894.3     0.1       0  5023.9    0.05       0  5027.9     0.1       0
Bank Sta=5023.9,5027.9
Exp/Cntr=0.3,0.1

Type RM Length L Ch R = 1,25417,530,530,530
BEGIN DESCRIPTION:
Bee Caves Creek 55.0
END DESCRIPTION:
XS GIS Cut Line= 4
      1815574.97     13916674.98      1815753.96     13916782.37
      1815890.06     13916759.94      1816124.98     13916525.02
#Sta/Elev= 30
  4763.8 2148.92  4787.2 2147.64  4835.7 2140.86  4894.1 2134.42  4962.1 2129.92
  4970.2 2127.21  4988.0 2126.44  5004.0 2121.10  5012.1 2121.08  5012.4 2120.58
  5016.1 2121.08  5034.4 2122.12  5044.0 2121.44  5054.7 2122.63  5074.9 2123.00
  5105.2 2123.11  5117.5 2121.99  5131.6 2123.71  5174.0 2125.71  5188.2 2127.09
  5195.2 2128.83  5202.3 2128.88  5244.7 2133.78  5258.9 2136.39  5273.0 2137.00
  5301.3 2140.46  5329.6 2144.38  5343.7 2147.56  5414.4 2153.25  5442.7 2156.26
#Mann=3,-1,0
  4763.8     0.1       0  5012.1    0.05       0  5016.1     0.1       0
Bank Sta=5012.1,5016.1
Exp/Cntr=0.3,0.1

Type RM Length L Ch R = 1,24887,482,482,482
BEGIN DESCRIPTION:
Bee Caves Creek 54.0
END DESCRIPTION:
XS GIS Cut Line= 3
      1815725.02     13917275.00      1816025.00     13917225.00
      1816174.99     13916925.02
#Sta/Elev= 30
  4695.9 2140.02  4756.7 2133.77  4784.6 2131.48  4789.7 2131.63  4807.4 2129.67
  4817.5 2128.10  4827.7 2125.68  4868.2 2120.30  4888.5 2119.27  4906.2 2116.95
  4939.2 2115.29  4959.5 2115.12  4967.1 2113.92  4989.9 2113.72  4997.5 2112.18
  5012.0 2112.06  5012.2 2111.56  5015.7 2111.56  5016.0 2112.06  5030.8 2112.70
  5036.3 2113.77  5044.7 2114.32  5053.1 2114.44  5058.7 2116.34  5096.5 2117.38
  5142.6 2120.25  5232.0 2129.06  5254.3 2130.53  5299.1 2134.24  5335.4 2136.36
#Mann=5,-1,0
  4695.9     0.1       0  5012.0    0.05       0  5016.0     0.1       0
  5096.5    0.07       0  5254.3     0.1       0
Bank Sta=5012,5016
Exp/Cntr=0.3,0.1

Type RM Length L Ch R = 1,24405,479,479,479
BEGIN DESCRIPTION:
Bee Caves Creek 53.0
END DESCRIPTION:
XS GIS Cut Line= 3
      1815825.01     13917525.00      1816125.00     13917675.00
      1816425.00     13917675.00
#Sta/Elev= 30
  4664.6 2126.39  4678.6 2124.93  4700.9 2124.26  4723.3 2121.88  4740.1 2121.16
  4768.0 2118.83  4784.8 2118.50  4807.1 2116.93  4829.5 2114.60  4896.6 2110.37
  4946.9 2109.43  4977.6 2109.60  4991.6 2108.83  4997.2 2107.13  5030.0 2107.56
  5038.0 2107.11  5038.3 2106.61  5041.8 2106.61  5042.0 2107.11  5050.0 2108.54
  5079.5 2110.06  5090.0 2110.55  5100.0 2109.91  5120.0 2111.42  5187.4 2114.39
  5200.0 2115.10  5230.0 2118.27  5260.0 2120.17  5280.0 2123.08  5300.0 2125.06
#Mann=5,-1,0
  4664.6     0.1       0  5038.0    0.05       0  5042.0     0.1       0
  5079.5    0.07       0  5187.4     0.1       0
Bank Sta=5038,5042
Exp/Cntr=0.3,0.1

Type RM Length L Ch R = 1,23926,423,423,423
BEGIN DESCRIPTION:
Bee Caves Creek 52.0
END DESCRIPTION:
XS GIS Cut Line= 3
      1815925.03     13918025.01      1816225.00     13918125.00
      1816525.03     13917824.97
#Sta/Elev= 30
  4690.2 2117.86  4721.8 2116.61  4742.9 2114.25  4785.0 2111.27  4795.6 2111.42
  4858.8 2108.38  4922.1 2106.43  4943.2 2105.33  4974.8 2102.03  4993.9 2101.95
  4994.1 2101.45  4997.6 2101.45  4997.9 2101.95  5003.8 2102.82  5034.7 2104.38
  5048.8 2104.52  5063.0 2103.30  5077.1 2104.69  5091.3 2104.82  5119.5 2103.63
  5133.7 2104.73  5204.4 2106.76  5232.7 2108.36  5261.0 2111.70  5275.1 2114.31
  5295.9 2119.12  5317.5 2123.45  5388.2 2129.99  5427.1 2135.42  5430.7 2135.42
#Mann=4,-1,0
  4690.2    0.07       0  4993.9    0.05       0  4997.9    0.07       0
  5295.9     0.1       0
Bank Sta=4993.9,4997.9
Exp/Cntr=0.3,0.1

Type RM Length L Ch R = 1,23503,474,474,474
BEGIN DESCRIPTION:
Bee Caves Creek 51.0
END DESCRIPTION:
XS GIS Cut Line= 3
      1816274.98     13918725.03      1816475.00     13918425.00
      1816775.03     13918124.97
#Sta/Elev= 30
  4634.3 2119.42  4637.3 2119.42  4641.8 2118.25  4647.9 2118.45  4662.9 2116.72
  4677.9 2113.84  4735.0 2109.74  4786.1 2103.76  4792.1 2102.40  4801.1 2101.97
  4828.1 2097.17  4837.1 2097.56  4850.7 2099.60  4864.2 2099.06  4879.2 2097.21
  4916.9 2099.48  4981.4 2100.39  4987.4 2099.42  5009.0 2099.19  5021.2 2097.16
  5021.4 2096.66  5025.2 2097.16  5037.3 2099.65  5051.5 2099.78  5108.0 2103.54
  5136.3 2104.49  5192.9 2108.45  5221.2 2109.24  5362.6 2117.83  5419.2 2124.23
#Mann=4,-1,0
  4634.3     0.1       0  4916.9    0.07       0  5021.2    0.05       0
  5025.2    0.07       0
Bank Sta=5021.2,5025.2
Exp/Cntr=0.3,0.1

Type RM Length L Ch R = 1,23029,442,442,442
BEGIN DESCRIPTION:
Bee Caves Creek 50.0
END DESCRIPTION:
XS GIS Cut Line= 3
      1816525.00     13918875.00      1816675.00     13918825.00
      1816986.63     13918511.99
#Sta/Elev= 30
  4841.9 2114.77  4852.4 2114.18  4863.0 2111.94  4884.1 2108.56  4894.6 2105.31
  4915.7 2101.11  4957.8 2094.47  4968.4 2091.87  4983.9 2087.35  4995.4 2083.93
  4995.6 2083.43  4999.1 2083.43  4999.4 2083.93  5003.5 2083.93  5007.1 2086.88
  5021.2 2088.45  5028.3 2088.57  5035.4 2090.69  5042.4 2090.44  5056.6 2092.16
  5155.6 2095.88  5198.0 2096.02  5226.3 2097.50  5233.4 2097.26  5314.2 2101.56
  5346.5 2102.36  5388.9 2105.24  5417.2 2106.08  5437.0 2107.75  5441.7 2107.75
#Mann=5,-1,0
  4841.9    0.07       0  4983.9     0.1       0  4995.4    0.05       0
  4999.4     0.1       0  5314.2    0.07       0
Bank Sta=4995.4,4999.4
Exp/Cntr=0.3,0.1

Type RM Length L Ch R = 1,22587,472,472,472
BEGIN DESCRIPTION:
Bee Caves Creek 49.0
END DESCRIPTION:
XS GIS Cut Line= 3
      1816874.99     13919225.01      1816925.00     13919175.00
      1817207.69     13918748.63
#Sta/Elev= 30
  4923.8 2089.31  4927.4 2089.31  4952.1 2086.44  4966.2 2083.88  4980.4 2078.78
  4989.0 2070.54  4989.2 2070.04  4992.7 2070.04  4993.0 2070.54  5008.1 2070.80
  5038.1 2072.86  5044.1 2075.91  5053.2 2078.59  5059.2 2081.15  5074.2 2083.62
  5089.3 2084.30  5095.3 2085.56  5138.5 2089.44  5188.5 2090.72  5233.7 2092.46
  5246.5 2092.34  5275.8 2093.21  5305.9 2094.68  5332.9 2094.95  5378.0 2097.48
  5405.1 2098.18  5441.2 2099.83  5471.3 2102.35  5503.2 2106.81  5506.1 2107.21
#Mann=4,-1,0
  4923.8     0.1       0  4989.0    0.05       0  4993.0     0.1       0
  5503.2    0.07       0
Bank Sta=4989,4993
Exp/Cntr=0.3,0.1

Type RM Length L Ch R = 1,22115,446,446,446
BEGIN DESCRIPTION:
Bee Caves Creek 48.0
END DESCRIPTION:
XS GIS Cut Line= 3
      1817175.00     13919625.00      1817225.00     13919525.00
      1817274.99     13919475.01
#Sta/Elev= 29
  4888.2 2091.01  4891.0 2091.01  4896.6 2090.12  4902.2 2089.36  4910.6 2087.54
  4918.9 2085.12  4924.5 2083.90  4932.9 2077.56  4935.0 2076.11  4941.3 2071.76
  4946.9 2067.35  4955.3 2064.50  4963.7 2063.22  4969.3 2062.40  4975.6 2062.27
  4975.9 2061.77  4979.4 2061.77  4979.6 2062.27  4986.0 2062.60  4991.6 2063.90
  4997.2 2066.24  5000.0 2066.24  5003.5 2066.24  5014.1 2067.85  5028.3 2069.92
  5042.4 2072.45  5056.6 2074.58  5067.2 2076.00  5070.7 2076.00
#Mann=4,-1,0
  4888.2     0.1       0  4935.0    0.07       0  4975.6    0.05       0
  4979.6    0.07       0
Bank Sta=4975.6,4979.6
Exp/Cntr=0.3,0.1

Type RM Length L Ch R = 1,21669,476,476,476
BEGIN DESCRIPTION:
Bee Caves Creek 47.0
END DESCRIPTION:
XS GIS Cut Line= 3
      1817575.00     13919825.00      1817575.00     13919775.00
      1817774.97     13919575.03
#Sta/Elev= 29
  4950.4 2078.25  4952.9 2078.25  4960.4 2077.90  4970.4 2076.77  4980.4 2075.09
  4990.4 2069.14  4997.9 2057.35  5003.9 2057.35  5012.4 2055.00  5012.7 2054.50
  5016.4 2054.50  5016.6 2055.00  5028.7 2055.05  5042.4 2057.00  5057.0 2058.80
  5071.1 2060.41  5085.3 2060.07  5099.4 2059.33  5127.7 2059.19  5141.8 2059.02
  5156.0 2063.59  5170.1 2068.69  5184.2 2072.32  5198.4 2075.82  5212.5 2078.62
  5226.7 2080.35  5269.1 2085.23  5279.7 2086.27  5283.2 2086.27
#Mann=4,-1,0
  4950.4     0.1       0  5012.4    0.05       0  5016.6     0.1       0
  5042.4     0.1       0
Bank Sta=5012.4,5016.6
Exp/Cntr=0.3,0.1

Type RM Length L Ch R = 1,21193,447,447,447
BEGIN DESCRIPTION:
Bee Caves Creek 46.0
END DESCRIPTION:
XS GIS Cut Line= 3
      1817575.01     13920374.99      1817975.00     13919975.00
      1818075.03     13919975.00
#Sta/Elev= 30
  4439.1 2117.94  4442.6 2117.94  4453.2 2114.02  4481.5 2109.38  4523.9 2100.04
  4545.1 2096.38  4580.5 2093.86  4608.8 2090.10  4637.1 2087.88  4665.4 2083.16
  4721.9 2076.75  4750.2 2072.34  4792.6 2062.26  4835.1 2056.45  4849.2 2054.90
  4863.3 2054.42  4934.1 2054.38  4948.2 2053.77  4962.3 2052.65  4976.5 2048.21
  4988.5 2047.97  4988.8 2047.47  4992.5 2047.47  4992.7 2047.97  5001.2 2063.07
  5007.3 2063.07  5014.8 2068.96  5024.8 2074.85  5034.8 2079.45  5104.8 2083.10
#Mann=3,-1,0
  4439.1     0.1       0  4988.5    0.05       0  4992.7     0.1       0
Bank Sta=4988.5,4992.7
Exp/Cntr=0.3,0.1

Type RM Length L Ch R = 1,20746,462,462,462
BEGIN DESCRIPTION:
Bee Caves Creek 45.0
END DESCRIPTION:
XS GIS Cut Line= 3
      1817974.98     13920525.02      1818125.00     13920375.00
      1818224.98     13920225.03
#Sta/Elev= 30
  4787.8 2084.37  4791.4 2084.37  4802.0 2082.32  4823.2 2080.83  4844.4 2074.74
  4872.7 2058.51  4886.8 2051.33  4901.0 2047.35  4915.1 2047.12  4929.2 2049.86
  4945.9 2050.20  4971.7 2048.97  4985.8 2045.20  4994.3 2044.80  4994.6 2044.30
  4998.3 2044.30  4998.6 2044.80  5003.0 2044.80  5013.5 2049.06  5022.5 2049.47
  5028.5 2050.75  5043.5 2051.45  5049.5 2052.41  5058.5 2055.54  5100.6 2060.32
  5115.6 2063.65  5120.4 2065.25  5151.7 2071.86  5157.7 2072.08  5180.2 2075.11
#Mann=5,-1,0
  4787.8     0.1       0  4945.9    0.07       0  4994.3    0.05       0
  4998.6    0.07       0  5120.4     0.1       0
Bank Sta=4994.3,4998.6
Exp/Cntr=0.3,0.1

Type RM Length L Ch R = 1,20284,460,460,460
BEGIN DESCRIPTION:
Bee Caves Creek 44.0
END DESCRIPTION:
XS GIS Cut Line= 3
      1818225.00     13920775.00      1818325.00     13920725.00
      1818475.00     13920325.00
#Sta/Elev= 30
  4888.4 2071.26  4891.2 2071.26  4933.1 2058.64  4963.9 2053.15  4987.0 2046.99
  4997.4 2041.04  5002.9 2041.04  5013.2 2037.27  5013.5 2036.77  5017.5 2037.27
  5021.6 2037.52  5040.3 2043.15  5085.6 2045.32  5095.4 2044.90  5100.8 2039.86
  5107.0 2038.25  5117.7 2039.70  5125.7 2043.41  5131.0 2042.32  5139.0 2046.71
  5148.2 2047.21  5156.0 2046.74  5186.2 2048.63  5192.4 2048.03  5216.5 2052.29
  5256.5 2056.36  5332.2 2060.81  5367.2 2066.84  5406.0 2072.55  5427.4 2073.92
#Mann=6,-1,0
  4888.4     0.1       0  4987.0    0.07       0  5013.2    0.05       0
  5017.5    0.07       0  5148.2     0.1       0  5367.2    0.07       0
Bank Sta=5013.2,5017.5
Exp/Cntr=0.3,0.1

Type RM Length L Ch R = 1,19824,465,465,465
BEGIN DESCRIPTION:
Bee Caves Creek 43.0
END DESCRIPTION:
XS GIS Cut Line= 3
      1818524.97     13921025.00      1818625.00     13921025.00
      1818974.97     13920925.01
#Sta/Elev= 30
  4900.3 2050.49  4940.3 2047.19  4950.3 2045.23  4960.3 2041.47  4980.3 2038.05
  4997.8 2032.79  5002.9 2032.79  5017.2 2036.31  5062.7 2037.88  5083.5 2037.26
  5095.2 2037.86  5114.7 2035.74  5126.9 2032.54  5127.2 2032.04  5130.9 2032.04
  5131.2 2032.54  5162.8 2039.11  5177.1 2039.03  5218.7 2041.32  5229.1 2040.63
  5235.6 2041.04  5249.9 2044.69  5260.3 2046.50  5269.4 2049.32  5281.1 2055.17
  5301.9 2060.93  5308.4 2064.58  5322.7 2069.77  5342.2 2074.44  5364.3 2076.04
#Mann=3,-1,0
  4900.3    0.07       0  5126.9    0.05       0  5131.2    0.07       0
Bank Sta=5126.9,5131.2
Exp/Cntr=0.3,0.1

Type RM Length L Ch R = 1,19359,449,449,449
BEGIN DESCRIPTION:
Bee Caves Creek 42.0
END DESCRIPTION:
XS GIS Cut Line= 3
      1818674.98     13921375.00      1818925.00     13921325.00
      1819125.02     13921224.99
#Sta/Elev= 30
  4740.8 2045.30  4781.6 2044.27  4802.0 2042.78  4822.4 2038.70  4842.8 2035.67
  4873.4 2033.53  4914.2 2035.42  4924.4 2034.08  4945.4 2035.63  4985.6 2034.42
  4993.2 2033.14  4998.6 2033.14  5004.2 2029.08  5006.8 2028.99  5007.3 2028.49
  5012.7 2028.99  5018.1 2030.44  5032.1 2032.30  5048.9 2032.72  5085.2 2035.74
  5093.6 2038.69  5099.2 2039.34  5105.7 2043.17  5116.0 2051.30  5121.6 2051.95
  5138.3 2058.40  5152.3 2061.34  5166.3 2066.07  5197.0 2078.96  5219.4 2080.75
#Mann=5,-1,0
  4740.8     0.1       0  4945.4    0.07       0  5006.8    0.05       0
  5012.7    0.07       0  5105.7     0.1       0
Bank Sta=5006.8,5012.7
Exp/Cntr=0.3,0.1

Type RM Length L Ch R = 1,18910,467,467,467
BEGIN DESCRIPTION:
Bee Caves Creek 41.0
END DESCRIPTION:
XS GIS Cut Line= 3
      1818724.95     13921674.99      1818975.00     13921725.00
      1819124.99     13921775.00
#Sta/Elev= 30
  4745.4 2043.62  4765.8 2043.05  4776.0 2042.24  4827.0 2035.79  4847.4 2031.62
  4857.6 2030.19  4867.8 2030.30  4878.0 2029.51  4895.2 2031.21  4939.2 2032.17
  4959.6 2030.04  4978.8 2028.77  4990.2 2028.41  4994.9 2026.18  4995.3 2025.68
  5000.3 2025.68  5000.8 2026.18  5010.9 2026.61  5032.0 2026.33  5042.6 2028.54
  5053.1 2032.82  5063.6 2039.13  5074.2 2048.41  5084.7 2053.09  5105.8 2060.85
  5126.9 2071.12  5137.4 2080.02  5148.0 2083.81  5155.9 2085.32  5158.5 2085.32
#Mann=5,-1,0
  4745.4     0.1       0  4895.2    0.07       0  4978.8     0.1       0
  4994.9    0.05       0  5000.8     0.1       0
Bank Sta=4994.9,5000.8
Exp/Cntr=0.3,0.1

Type RM Length L Ch R = 1,18443,479,479,479
BEGIN DESCRIPTION:
Bee Caves Creek 40.0
END DESCRIPTION:
XS GIS Cut Line= 3
      1818625.02     13922175.00      1818925.00     13922175.00
      1819125.02     13922175.00
#Sta/Elev= 30
  4700.1 2046.12  4740.1 2045.38  4750.1 2043.99  4800.1 2032.72  4820.1 2026.54
  4840.1 2025.55  4847.1 2024.12  4847.6 2023.62  4852.6 2023.62  4853.1 2024.12
  4870.1 2025.53  4880.1 2025.25  4890.1 2024.22  4920.1 2026.05  4930.1 2026.12
  4950.1 2025.34  4970.1 2025.94  5010.1 2024.16  5020.1 2025.07  5030.1 2026.76
  5040.1 2031.63  5050.1 2039.06  5060.1 2043.92  5080.1 2050.91  5110.1 2059.60
  5140.1 2070.62  5150.1 2079.69  5160.1 2083.41  5170.1 2084.94  5200.1 2087.30
#Mann=3,-1,0
  4700.1     0.1       0  4847.1    0.05       0  4853.1     0.1       0
Bank Sta=4847.1,4853.1
Exp/Cntr=0.3,0.1

Type RM Length L Ch R = 1,17964,484,484,484
BEGIN DESCRIPTION:
Bee Caves Creek 39.0
END DESCRIPTION:
XS GIS Cut Line= 3
      1818575.04     13922475.02      1818825.00     13922625.00
      1819124.97     13922525.01
#Sta/Elev= 30
  4702.7 2045.21  4737.6 2042.65  4747.4 2040.03  4753.2 2039.48  4774.6 2034.55
  4795.9 2027.02  4805.7 2021.87  4819.3 2019.84  4827.0 2020.20  4832.9 2021.86
  4854.0 2021.80  4922.3 2023.76  4949.5 2021.96  4975.7 2023.68  4996.8 2022.91
  5022.8 2018.81  5023.3 2018.31  5028.8 2018.81  5046.9 2020.59  5057.4 2022.93
  5120.7 2041.58  5141.8 2046.81  5162.9 2050.05  5215.6 2055.93  5236.6 2060.21
  5257.7 2065.70  5268.3 2070.67  5278.8 2073.10  5299.9 2075.49  5310.4 2075.69
#Mann=5,-1,0
  4702.7     0.1       0  4854.0    0.07       0  4975.7     0.1       0
  5022.8    0.05       0  5028.8     0.1       0
Bank Sta=5022.8,5028.8
Exp/Cntr=0.3,0.1

Type RM Length L Ch R = 1,17480,467,467,467
BEGIN DESCRIPTION:
Bee Caves Creek 38.0
END DESCRIPTION:
XS GIS Cut Line= 3
      1818324.97     13923225.01      1818725.00     13923075.00
      1818874.97     13923075.00
#Sta/Elev= 30
  4568.2 2077.41  4613.6 2075.42  4632.3 2068.74  4638.5 2065.38  4643.9 2064.62
  4663.5 2057.68  4707.1 2050.06  4724.0 2045.24  4729.3 2045.40  4742.5 2040.97
  4748.9 2037.56  4754.2 2038.49  4760.5 2034.20  4779.2 2027.04  4784.5 2027.80
  4809.4 2020.22  4814.8 2020.67  4849.1 2017.28  4878.0 2016.80  4894.9 2018.73
  4942.0 2016.95  4985.6 2017.06  5011.9 2014.29  5012.4 2013.79  5018.9 2014.29
  5035.4 2018.00  5055.4 2024.47  5092.6 2030.70  5124.1 2033.87  5145.4 2036.12
#Mann=7,-1,0
  4568.2     0.1       0  4742.5    0.07       0  4849.1     0.1       0
  5011.9    0.05       0  5018.9     0.1       0  5092.6    0.07       0
  5124.1     0.1       0
Bank Sta=5011.9,5018.9
Exp/Cntr=0.3,0.1

Type RM Length L Ch R = 1,17013,485,485,485
BEGIN DESCRIPTION:
Bee Caves Creek 37.0
END DESCRIPTION:
XS GIS Cut Line= 3
      1818375.02     13923425.01      1818775.00     13923525.00
      1818874.99     13923425.01
#Sta/Elev= 30
  4587.7 2060.74  4646.9 2050.75  4652.1 2051.09  4680.4 2045.58  4688.2 2042.00
  4693.3 2042.25  4701.1 2037.45  4721.7 2029.83  4729.4 2025.17  4734.6 2025.95
  4742.3 2021.41  4752.6 2019.11  4770.6 2017.56  4811.9 2018.55  4853.1 2016.75
  4876.3 2018.35  4899.5 2017.42  4917.5 2014.97  4940.7 2014.44  4948.3 2013.00
  4969.1 2013.55  4976.8 2011.07  4982.0 2011.36  4986.1 2010.10  4986.6 2009.60
  4993.2 2010.10  5003.5 2010.60  5042.4 2020.78  5123.7 2025.72  5141.4 2027.19
#Mann=5,-1,0
  4587.7     0.1       0  4948.3    0.07       0  4986.1    0.05       0
  4993.2    0.07       0  5123.7     0.1       0
Bank Sta=4986.1,4993.2
Exp/Cntr=0.3,0.1

Type RM Length L Ch R = 1,16528,479,479,479
BEGIN DESCRIPTION:
Bee Caves Creek 36.0
END DESCRIPTION:
XS GIS Cut Line= 3
      1818775.03     13924074.97      1818875.00     13923975.00
      1819225.01     13923574.99
#Sta/Elev= 30
  4863.7 2046.65  4891.9 2044.50  4906.1 2042.27  4920.2 2038.38  4934.4 2030.14
  4948.5 2018.75  4962.7 2009.94  4973.1 2007.18  4973.6 2006.68  4980.5 2007.18
  5001.5 2010.05  5012.2 2009.99  5018.8 2010.94  5033.1 2010.56  5090.0 2012.26
  5118.5 2014.24  5217.7 2014.57  5231.4 2011.60  5245.7 2010.68  5253.3 2012.59
  5274.2 2012.31  5288.4 2013.33  5296.0 2015.09  5316.9 2016.62  5345.3 2021.83
  5366.2 2023.67  5402.3 2028.47  5472.5 2033.31  5508.6 2037.41  5536.6 2039.35
#Mann=3,-1,0
  4863.7     0.1       0  4973.1    0.05       0  4980.5     0.1       0
Bank Sta=4973.1,4980.5
Exp/Cntr=0.3,0.1

Type RM Length L Ch R = 1,16049,450,450,450
BEGIN DESCRIPTION:
Bee Caves Creek 35.0
END DESCRIPTION:
XS GIS Cut Line= 3
      1819275.00     13924325.02      1819275.00     13924125.00
      1819374.99     13923725.03
#Sta/Elev= 30
  4800.0 2081.38  4820.0 2077.97  4840.0 2066.66  4880.0 2047.69  4890.0 2042.42
  4920.0 2022.87  4930.0 2015.44  4940.0 2009.98  4950.0 2006.91  4960.0 2005.23
  4980.0 2004.11  4993.8 2001.81  4994.3 2001.31  5000.8 2001.31  5001.3 2001.81
  5010.3 2003.87  5018.1 2007.30  5041.2 2007.43  5059.3 2008.98  5100.5 2009.42
  5113.4 2008.98  5183.0 2010.60  5216.5 2009.66  5229.4 2010.90  5237.1 2010.93
  5247.4 2010.22  5257.7 2007.98  5329.9 2019.81  5371.1 2025.26  5412.3 2028.97
#Mann=3,-1,0
  4800.0     0.1       0  4993.8    0.05       0  5001.3     0.1       0
Bank Sta=4993.8,5001.3
Exp/Cntr=0.3,0.1

Type RM Length L Ch R = 1,15599,458,458,458
BEGIN DESCRIPTION:
Bee Caves Creek 34.0
END DESCRIPTION:
XS GIS Cut Line= 3
      1819574.98     13924375.03      1819725.00     13924125.00
      1819825.00     13923725.00
#Sta/Elev= 30
  4708.9 2081.29  4732.3 2079.29  4743.9 2073.25  4759.5 2067.88  4775.0 2061.00
  4817.8 2050.55  4833.3 2042.96  4839.2 2042.27  4870.3 2027.50  4876.1 2026.10
  4891.6 2016.52  4897.5 2015.90  4907.2 2012.05  4928.6 2005.98  4965.5 2002.80
  4986.9 2003.31  5007.0 2001.95  5007.5 2001.45  5014.6 2001.95  5031.4 2003.60
  5041.7 2002.81  5082.9 2004.93  5124.2 2004.00  5142.2 2006.44  5147.4 2006.02
  5183.5 2011.45  5188.6 2011.24  5289.1 2021.97  5312.3 2023.40  5412.8 2033.04
#Mann=3,-1,0
  4708.9     0.1       0  5007.0    0.05       0  5014.6     0.1       0
Bank Sta=5007,5014.6
Exp/Cntr=0.3,0.1

Type RM Length L Ch R = 1,15141,466,466,466
BEGIN DESCRIPTION:
Bee Caves Creek 33.0
END DESCRIPTION:
XS GIS Cut Line= 3
      1819925.00     13924375.00      1820125.00     13923975.00
      1820125.00     13923875.02
#Sta/Elev= 30
  4552.4 2043.26  4627.9 2026.15  4633.5 2026.08  4650.2 2020.88  4655.8 2020.83
  4686.6 2013.55  4700.5 2012.08  4717.3 2007.73  4722.9 2007.38  4731.3 2001.83
  4745.3 2000.78  4806.8 2001.65  4829.1 2003.65  4843.1 2003.23  4851.5 1999.99
  4857.1 1999.51  4865.5 1999.77  4873.8 2002.60  4887.8 2003.03  4918.6 2002.12
  4954.9 1998.93  4968.9 1999.37  4987.4 1997.99  4987.9 1997.49  4995.1 1997.99
  4996.8 1999.86  5002.1 1999.86  5019.6 2008.12  5029.6 2010.60  5099.6 2020.71
#Mann=3,-1,0
  4552.4     0.1       0  4987.4    0.05       0  4995.1     0.1       0
Bank Sta=4987.4,4995.1
Exp/Cntr=0.3,0.1

Type RM Length L Ch R = 1,14675,448,448,448
BEGIN DESCRIPTION:
Bee Caves Creek 32.0
END DESCRIPTION:
XS GIS Cut Line= 3
      1820275.00     13924425.00      1820575.00     13924025.00
      1820625.00     13923925.01
#Sta/Elev= 30
  4499.9 2024.00  4671.8 2009.06  4713.4 2006.98  4742.6 2003.50  4757.2 1999.37
  4771.8 1998.30  4821.8 1999.26  4842.6 1998.44  4878.0 2000.17  4907.2 1997.32
  4913.4 1998.40  4936.4 1997.05  4942.6 1997.91  4957.2 1996.49  4978.0 1996.99
  4992.6 1996.06  4996.8 1994.38  5002.7 1994.38  5010.0 1992.08  5010.5 1991.58
  5017.7 1992.08  5022.3 1995.04  5036.2 1997.51  5044.6 2003.27  5053.0 2012.10
  5058.6 2014.04  5075.4 2022.68  5081.0 2022.98  5097.7 2028.86  5111.7 2030.86
#Mann=3,-1,0
  4499.9     0.1       0  5010.0    0.05       0  5017.7     0.1       0
Bank Sta=5010,5017.7
Exp/Cntr=0.3,0.1

Type RM Length L Ch R = 1,14227,469,469,469
BEGIN DESCRIPTION:
Bee Caves Creek 31.0
END DESCRIPTION:
XS GIS Cut Line= 3
      1820575.00     13924575.00      1820975.00     13924175.00
      1820975.00     13924074.99
#Sta/Elev= 30
  4434.4 2018.55  4491.0 2016.06  4533.4 2012.93  4561.7 2011.86  4674.8 2004.96
  4703.1 2004.35  4745.5 2000.75  4778.1 1998.93  4802.1 1998.13  4829.9 1998.23
  4844.5 1997.70  4872.8 1998.52  4901.1 1997.95  4922.2 1995.54  4943.5 1993.32
  4957.7 1994.63  4971.8 1994.43  4981.2 1991.08  4992.7 1987.58  4993.2 1987.08
  5000.0 1987.08  5000.5 1987.58  5010.1 1988.20  5020.1 1990.04  5030.1 1994.09
  5040.1 2001.13  5050.1 2009.28  5070.1 2015.11  5097.6 2021.03  5100.1 2021.03
#Mann=7,-1,0
  4434.4     0.1       0  4778.1    0.07       0  4829.9     0.1       0
  4922.2    0.07       0  4981.2     0.1       0  4992.7    0.05       0
  5000.5     0.1       0
Bank Sta=4992.7,5000.5
Exp/Cntr=0.3,0.1

Type RM Length L Ch R = 1,13758,453,453,453
BEGIN DESCRIPTION:
Bee Caves Creek 30.0
END DESCRIPTION:
XS GIS Cut Line= 3
      1820875.04     13924674.98      1821275.00     13924475.00
      1821625.02     13924575.01
#Sta/Elev= 30
  4552.5 2008.36  4717.4 1996.56  4843.1 1990.81  4932.6 1991.72  4946.6 1991.09
  4963.3 1987.90  4980.2 1986.40  4980.7 1985.90  4991.1 1986.40  5016.6 1987.94
  5021.8 1986.94  5050.4 1992.36  5072.5 1994.42  5134.9 1994.44  5155.7 1996.31
  5162.2 1998.39  5167.4 1996.97  5176.5 1998.92  5196.0 2006.10  5201.2 2003.69
  5207.7 2010.08  5228.5 2017.10  5235.0 2020.81  5240.2 2020.36  5259.7 2027.99
  5268.8 2030.30  5274.0 2030.10  5280.5 2032.59  5341.6 2046.28  5363.7 2049.56
#Mann=3,-1,0
  4552.5    0.07       0  4980.2    0.05       0  4991.1     0.1       0
Bank Sta=4980.2,4991.1
Exp/Cntr=0.3,0.1

Type RM Length L Ch R = 1,13305,453,453,453
BEGIN DESCRIPTION:
Bee Caves Creek 29.0
END DESCRIPTION:
XS GIS Cut Line= 3
      1820725.00     13924775.00      1821425.00     13924875.00
      1821625.00     13924725.00
#Sta/Elev= 30
  4292.3 2016.28  4368.7 2012.79  4514.5 2005.54  4656.0 1993.30  4676.2 1990.67
  4686.3 1987.20  4736.8 1986.80  4764.0 1989.35  4787.3 1990.47  4847.9 1988.08
  4868.1 1990.30  4948.9 1989.61  5015.8 1984.77  5016.3 1984.27  5026.7 1984.77
  5042.1 1988.65  5099.4 1990.31  5121.3 1995.72  5127.5 1995.54  5135.9 1999.84
  5142.1 2000.18  5156.7 2012.71  5162.9 2011.04  5171.3 2017.16  5177.5 2017.03
  5185.9 2022.26  5192.1 2022.47  5206.7 2034.55  5221.3 2040.87  5249.4 2045.87
#Mann=5,-1,0
  4292.3     0.1       0  4368.7    0.07       0  4764.0     0.1       0
  5015.8    0.05       0  5026.7     0.1       0
Bank Sta=5015.8,5026.7
Exp/Cntr=0.3,0.1

Type RM Length L Ch R = 1,12852,519,519,519
BEGIN DESCRIPTION:
Bee Caves Creek 28.0
END DESCRIPTION:
XS GIS Cut Line= 3
      1820824.97     13924924.97      1821175.00     13925225.00
      1821274.98     13925274.99
#Sta/Elev= 30
  4544.0 2008.81  4565.4 2007.81  4671.9 1999.50  4716.3 1994.75  4735.6 1991.57
  4770.7 1989.02  4792.6 1985.54  4799.2 1985.31  4820.6 1980.95  4834.3 1980.18
  4842.0 1980.32  4856.3 1982.90  4877.2 1981.65  4899.1 1985.43  4921.3 1985.58
  4948.5 1985.95  4978.1 1979.77  4978.6 1979.27  4989.1 1979.77  4997.9 1981.17
  5001.7 1983.30  5007.8 1983.30  5013.4 1986.05  5019.0 1991.54  5035.8 1998.96
  5041.4 2002.54  5058.1 2009.52  5102.8 2018.12  5108.4 2017.93  5116.8 2019.32
#Mann=5,-1,0
  4544.0     0.1       0  4716.3    0.07       0  4921.3     0.1       0
  4978.1    0.05       0  4989.1     0.1       0
Bank Sta=4978.1,4989.1
Exp/Cntr=0.3,0.1

Type RM Length L Ch R = 1,12333,374,374,374
BEGIN DESCRIPTION:
Bee Caves Creek 27.0
END DESCRIPTION:
XS GIS Cut Line= 3
      1820475.00     13925325.00      1820843.44     13925543.34
      1821174.95     13925525.00
#Sta/Elev= 30
  4635.6 2023.66  4693.7 2017.97  4738.9 2011.83  4744.8 2011.83  4760.4 2007.66
  4818.9 1998.16  4861.7 1989.91  4883.2 1984.63  4923.3 1982.87  4963.1 1981.99
  4978.7 1978.76  4990.3 1978.19  5007.6 1976.69  5025.2 1976.63  5025.7 1976.13
  5036.4 1976.63  5052.8 1977.08  5061.9 1978.51  5075.5 1978.06  5085.5 1979.31
  5115.5 1979.85  5122.5 1982.30  5127.5 1980.79  5145.6 1985.99  5185.6 1990.44
  5235.7 1993.40  5303.1 2002.11  5335.9 2005.21  5375.9 2010.97  5395.9 2012.51
#Mann=5,-1,0
  4635.6     0.1       0  4923.3    0.07       0  4990.3     0.1       0
  5025.2    0.05       0  5036.4     0.1       0
Bank Sta=5025.2,5036.4
Exp/Cntr=0.3,0.1

Type RM Length L Ch R = 1,11959,461,461,461
BEGIN DESCRIPTION:
Bee Caves Creek 26.0
END DESCRIPTION:
XS GIS Cut Line= 3
      1820224.98     13925724.99      1820625.00     13925825.00
      1820875.02     13925975.01
#Sta/Elev= 30
  4591.9 2062.48  4610.0 2058.72  4615.1 2058.64  4651.2 2048.94  4656.3 2048.70
  4684.7 2039.81  4692.4 2035.29  4697.6 2033.98  4715.6 2025.36  4733.7 2013.84
  4738.8 2011.81  4746.5 2005.27  4756.8 1998.72  4774.9 1988.99  4787.8 1983.95
  4816.1 1980.15  4880.5 1977.99  4963.0 1979.90  4973.3 1978.28  4980.6 1973.40
  4981.1 1972.90  4991.8 1973.40  5027.6 1975.88  5113.1 1977.07  5144.2 1981.33
  5155.8 1984.85  5171.3 1986.84  5186.9 1989.52  5278.9 1999.64  5295.8 2000.37
#Mann=5,-1,0
  4591.9     0.1       0  4980.6    0.05       0  4991.8     0.1       0
  5171.3    0.07       0  5278.9     0.1       0
Bank Sta=4980.6,4991.8
Exp/Cntr=0.3,0.1

Type RM Length L Ch R = 1,11498,482,482,482
BEGIN DESCRIPTION:
Bee Caves Creek 25.0
END DESCRIPTION:
XS GIS Cut Line= 3
      1820225.02     13926324.99      1820525.00     13926225.00
      1820824.96     13926175.01
#Sta/Elev= 30
  4683.9 2067.63  4705.0 2063.83  4715.5 2060.47  4747.1 2029.16  4757.7 2022.70
  4768.2 2014.52  4789.3 2003.63  4799.8 1996.14  4831.4 1983.88  4842.0 1982.02
  4863.1 1973.45  4915.8 1974.19  4926.3 1971.68  4936.9 1971.58  4968.5 1973.37
  5002.6 1971.48  5004.6 1970.02  5005.1 1969.52  5015.8 1970.02  5033.1 1971.64
  5050.8 1975.68  5071.1 1977.01  5135.5 1974.04  5142.0 1974.77  5149.6 1978.43
  5154.7 1977.99  5162.3 1982.41  5172.4 1985.71  5282.6 1996.69  5304.2 1998.52
#Mann=5,-1,0
  4683.9     0.1       0  5004.6    0.05       0  5015.8     0.1       0
  5135.5    0.07       0  5282.6     0.1       0
Bank Sta=5004.6,5015.8
Exp/Cntr=0.3,0.1

Type RM Length L Ch R = 1,11016,539,539,539
BEGIN DESCRIPTION:
Bee Caves Creek 24.0
END DESCRIPTION:
XS GIS Cut Line= 3
      1820524.96     13926725.02      1820625.00     13926675.00
      1820924.99     13926375.01
#Sta/Elev= 30
  4880.2 2037.51  4883.0 2037.51  4888.6 2035.79  4894.2 2035.67  4916.6 2028.84
  4947.3 2012.67  4955.7 2005.97  4961.3 2000.63  4969.7 1995.43  4978.1 1991.19
  4983.7 1986.86  4989.3 1981.05  4995.6 1981.05  5000.5 1965.59  5001.0 1965.09
  5011.8 1965.59  5020.3 1967.09  5048.6 1968.47  5064.5 1970.20  5091.0 1970.25
  5133.5 1971.80  5158.7 1973.49  5218.3 1977.24  5232.5 1978.76  5260.8 1983.63
  5289.0 1986.06  5317.3 1989.73  5331.5 1990.09  5402.2 1995.97  5416.3 1996.51
#Mann=5,-1,0
  4880.2     0.1       0  5000.5    0.05       0  5011.8     0.1       0
  5064.5    0.07       0  5158.7     0.1       0
Bank Sta=5000.5,5011.8
Exp/Cntr=0.3,0.1

Type RM Length L Ch R = 1,10477,458,458,458
BEGIN DESCRIPTION:
Bee Caves Creek 23.0
END DESCRIPTION:
XS GIS Cut Line= 3
      1820846.29     13926989.43      1821058.15     13926931.57
      1821174.98     13926675.04
#Sta/Elev= 30
  4801.8 1995.48  4810.8 1993.49  4837.2 1990.18  4862.7 1987.66  4876.9 1985.13
  4904.1 1978.04  4911.4 1975.72  4916.6 1970.78  4924.9 1966.16  4935.2 1964.10
  4968.6 1965.25  4985.7 1964.87  4990.6 1964.13  4997.4 1963.19  5007.8 1962.74
  5070.6 1962.93  5076.1 1962.38  5093.5 1962.01  5094.0 1961.51  5104.3 1961.51
  5104.8 1962.01  5138.5 1967.41  5145.3 1969.36  5150.8 1970.27  5168.3 1971.20
  5191.4 1973.69  5214.4 1979.14  5237.4 1983.25  5281.4 1988.72  5303.3 1989.38
#Mann=5,-1,0
  4801.8     0.1       0  4968.6    0.07       0  4990.6     0.1       0
  5093.5    0.05       0  5104.8     0.1       0
Bank Sta=5093.5,5104.8
Exp/Cntr=0.3,0.1

Type RM Length L Ch R = 1,10019,374,374,374
BEGIN DESCRIPTION:
Bee Caves Creek 22.0
END DESCRIPTION:
XS GIS Cut Line= 3
      1821184.65     13927282.47      1821400.57     13927103.28
      1821799.76     13927032.53
#Sta/Elev= 30
  4716.7 1985.20  4736.4 1983.76  4849.7 1979.63  4899.2 1971.05  4907.0 1969.33
  4913.5 1965.83  4923.2 1963.48  4927.9 1962.68  4935.7 1963.34  4990.9 1960.38
  4991.4 1959.88  5002.9 1960.38  5022.1 1961.95  5042.4 1962.12  5062.7 1963.91
  5070.6 1963.31  5075.7 1966.40  5093.2 1966.85  5113.5 1968.94  5123.7 1970.72
  5144.0 1979.14  5165.9 1986.80  5174.4 1989.40  5225.2 1998.94  5296.3 2008.25
  5302.0 2009.86  5316.6 2009.70  5347.1 2013.28  5361.1 2013.46  5402.7 2017.00
#Mann=5,-1,0
  4716.7     0.1       0  4923.2    0.07       0  4990.9    0.05       0
  5002.9    0.07       0  5165.9     0.1       0
Bank Sta=4990.9,5002.9
Exp/Cntr=0.3,0.1

Type RM Length L Ch R = 1,9645,435,435,435
BEGIN DESCRIPTION:
Bee Caves Creek 21.0
END DESCRIPTION:
XS GIS Cut Line= 3
      1821274.98     13927525.01      1821675.00     13927325.00
      1821824.95     13927275.02
#Sta/Elev= 30
  4552.7 1986.27  4587.2 1983.80  4611.4 1981.89  4650.5 1976.08  4696.5 1972.00
  4698.8 1971.79  4745.6 1968.65  4762.4 1966.59  4790.3 1965.64  4798.7 1964.00
  4829.4 1966.54  4857.4 1967.29  4918.9 1965.49  4941.2 1963.21  4969.2 1961.75
  4986.0 1958.74  4991.5 1956.96  5002.6 1956.08  5004.5 1954.86  5005.0 1954.36
  5016.5 1954.86  5031.6 1956.54  5042.1 1961.92  5052.6 1978.80  5063.2 1986.32
  5073.7 1991.93  5084.3 1999.30  5115.9 2013.71  5147.5 2023.72  5158.0 2024.77
#Mann=6,-1,0
  4552.7    0.07       0  4587.2     0.1       0  4696.5    0.07       0
  4698.8     0.1       0  5004.5    0.05       0  5016.5     0.1       0
Bank Sta=5004.5,5016.5
Exp/Cntr=0.3,0.1

Type RM Length L Ch R = 1,9210,487,487,487
BEGIN DESCRIPTION:
Bee Caves Creek 20.0
END DESCRIPTION:
XS GIS Cut Line= 3
      1821425.04     13927774.99      1821675.00     13927725.00
      1821974.99     13927725.00
#Sta/Elev= 30
  4745.5 1982.13  4796.4 1976.59  4837.2 1970.05  4857.6 1965.66  4867.8 1964.05
  4908.6 1961.73  4929.0 1959.46  4959.6 1958.55  4990.2 1953.99  5014.4 1953.49
  5014.9 1952.99  5025.9 1952.99  5026.4 1953.49  5030.4 1955.31  5040.4 1955.96
  5050.4 1959.76  5060.4 1966.23  5070.4 1971.69  5090.4 1980.14  5100.4 1983.33
  5110.4 1987.87  5120.4 1991.26  5130.4 1993.41  5140.4 1997.47  5200.4 2015.64
  5230.4 2026.64  5250.4 2031.96  5280.4 2041.69  5297.9 2046.77  5300.4 2046.77
#Mann=3,-1,0
  4745.5     0.1       0  5014.4    0.05       0  5026.4     0.1       0
Bank Sta=5014.4,5026.4
Exp/Cntr=0.3,0.1

Type RM Length L Ch R = 1,8723,450,450,450
BEGIN DESCRIPTION:
Bee Caves Creek 19.0
END DESCRIPTION:
XS GIS Cut Line= 3
      1821424.99     13928075.00      1821575.00     13928175.00
      1821775.01     13928325.01
#Sta/Elev= 30
  4819.7 1973.22  4842.2 1970.34  4869.3 1968.27  4891.8 1963.53  4899.3 1960.68
  4914.4 1958.31  4941.4 1958.69  4950.4 1954.92  4956.4 1954.79  4965.4 1949.84
  4965.9 1949.34  4977.4 1949.84  4992.5 1951.45  4997.0 1953.00  5006.1 1953.32
  5021.9 1954.20  5050.0 1953.78  5071.9 1955.85  5086.4 1955.51  5113.5 1952.28
  5128.1 1952.16  5136.4 1954.83  5142.7 1960.19  5150.0 1969.22  5157.3 1976.82
  5163.5 1982.30  5171.9 1987.16  5192.7 1992.45  5207.3 1998.43  5250.0 2006.63
#Mann=4,-1,0
  4819.7     0.1       0  4965.4    0.05       0  4977.4     0.1       0
  5006.1    0.07       0
Bank Sta=4965.4,4977.4
Exp/Cntr=0.3,0.1

Type RM Length L Ch R = 1,8273,444,444,444
BEGIN DESCRIPTION:
Bee Caves Creek 18.0
END DESCRIPTION:
XS GIS Cut Line= 3
      1821025.02     13928275.01      1821425.00     13928575.00
      1821525.02     13928625.01
#Sta/Elev= 30
  4499.8 1991.60  4527.9 1990.08  4542.5 1987.86  4557.1 1987.12  4571.7 1985.28
  4577.9 1982.85  4586.2 1981.90  4592.5 1979.90  4654.2 1970.08  4686.2 1965.80
  4707.1 1962.07  4763.3 1956.44  4827.9 1954.92  4849.8 1955.20  4863.3 1954.03
  4886.2 1954.92  4921.7 1954.58  4957.1 1947.28  4971.7 1948.39  5002.6 1946.94
  5007.7 1946.23  5008.2 1945.73  5019.3 1945.73  5019.8 1946.23  5045.1 1950.11
  5052.9 1953.75  5058.5 1977.82  5066.9 1981.50  5097.6 1985.86  5111.6 1987.09
#Mann=5,-1,0
  4499.8     0.1       0  4654.2    0.07       0  5007.7    0.05       0
  5019.8    0.07       0  5045.1     0.1       0
Bank Sta=5007.7,5019.8
Exp/Cntr=0.3,0.1

Type RM Length L Ch R = 1,7829,475,475,475
BEGIN DESCRIPTION:
Bee Caves Creek 17.0
END DESCRIPTION:
XS GIS Cut Line= 3
      1820775.00     13928825.00      1821075.00     13928825.00
      1821225.00     13928825.00
#Sta/Elev= 30
  4700.3 1995.93  4702.8 1995.93  4730.3 1991.99  4740.3 1988.19  4750.3 1975.59
  4760.3 1966.63  4780.3 1957.30  4790.3 1954.36  4800.3 1952.75  4820.3 1950.77
  4870.3 1948.00  4893.0 1946.14  4910.3 1945.33  4920.3 1943.73  4939.5 1943.50
  4944.3 1943.10  4944.8 1942.60  4955.9 1942.60  4956.4 1943.10  4991.5 1944.09
  5010.3 1943.97  5030.3 1944.88  5040.3 1947.17  5050.3 1950.29  5070.3 1954.93
  5092.4 1958.22  5119.0 1962.53  5130.3 1963.84  5147.8 1967.29  5150.3 1967.29
#Mann=8,-1,0
  4700.3    0.07       0  4893.0   0.035       0  4939.5    0.07       0
  4944.3   0.035       0  4956.4    0.07       0  4991.5   0.035       0
  5092.4    0.07       0  5119.0     0.1       0
Bank Sta=4944.3,4956.4
Exp/Cntr=0.3,0.1

Type RM Length L Ch R = 1,7354,447,447,447
BEGIN DESCRIPTION:
Bee Caves Creek 16.0
END DESCRIPTION:
XS GIS Cut Line= 3
      1820875.00     13929125.00      1820975.00     13929225.00
      1821374.97     13929175.00
#Sta/Elev= 30
  4853.8 1972.30  4857.3 1972.30  4867.9 1970.35  4896.2 1966.75  4924.5 1961.99
  4936.2 1954.94  4952.8 1946.61  4966.9 1942.27  4981.1 1939.18  4991.7 1937.93
  5005.3 1938.46  5009.2 1936.87  5009.7 1936.37  5021.1 1936.37  5021.6 1936.87
  5033.0 1939.78  5038.0 1940.16  5045.6 1943.52  5064.8 1945.32  5103.7 1948.35
  5126.2 1950.13  5199.3 1952.11  5222.7 1953.90  5229.8 1954.72  5257.2 1959.65
  5274.9 1963.58  5279.9 1963.73  5355.5 1975.57  5360.5 1975.59  5398.3 1979.49
#Mann=8,-1,0
  4853.8     0.1       0  4936.2    0.07       0  5009.2    0.05       0
  5021.6    0.07       0  5064.8     0.1       0  5103.7    0.07       0
  5222.7     0.1       0  5229.8    0.07       0
Bank Sta=5009.2,5021.6
Exp/Cntr=0.3,0.1

Type RM Length L Ch R = 1,6907,457,457,457
BEGIN DESCRIPTION:
Bee Caves Creek 15.0
END DESCRIPTION:
XS GIS Cut Line= 3
      1820825.02     13929625.00      1821125.00     13929625.00
      1821374.97     13929575.01
#Sta/Elev= 30
  4705.1 1986.42  4725.1 1984.47  4735.1 1981.75  4755.1 1974.56  4775.1 1968.13
  4795.1 1962.89  4815.1 1958.80  4825.1 1956.05  4875.1 1947.63  4915.1 1942.59
  4945.1 1940.38  4955.1 1938.75  4978.8 1937.17  4979.3 1936.67  4990.8 1936.67
  4991.3 1937.17  5015.3 1937.30  5025.5 1938.12  5056.1 1938.95  5076.5 1940.74
  5086.7 1943.54  5096.9 1944.77  5127.5 1945.82  5158.0 1948.61  5168.2 1950.84
  5178.4 1954.51  5188.6 1959.86  5198.8 1966.91  5209.0 1969.45  5260.0 1973.93
#Mann=3,-1,0
  4705.1    0.07       0  4978.8    0.05       0  4991.3     0.1       0
Bank Sta=4978.8,4991.3
Exp/Cntr=0.3,0.1

Type RM Length L Ch R = 1,6450,450,450,450
BEGIN DESCRIPTION:
Bee Caves Creek 14.0
END DESCRIPTION:
XS GIS Cut Line= 3
      1820975.01     13930174.99      1821275.00     13930025.00
      1821475.01     13929875.00
#Sta/Elev= 30
  4664.6 1996.36  4695.3 1993.67  4717.7 1988.47  4731.7 1982.96  4739.3 1977.48
  4745.6 1971.93  4754.0 1966.01  4762.4 1957.46  4784.8 1946.56  4807.1 1944.19
  4821.1 1944.47  4874.2 1942.38  4879.8 1941.55  4888.2 1938.87  4896.6 1935.03
  4902.2 1935.48  4924.5 1934.14  4946.9 1934.89  4963.7 1934.13  4969.2 1935.14
  4990.9 1933.38  4991.4 1932.88  5003.4 1933.38  5007.3 1935.04  5042.7 1938.40
  5078.1 1944.54  5121.9 1949.32  5200.0 1960.88  5228.1 1963.11  5250.0 1966.12
#Mann=4,-1,0
  4664.6     0.1       0  4739.3    0.07       0  4990.9    0.05       0
  5003.4     0.1       0
Bank Sta=4990.9,5003.4
Exp/Cntr=0.3,0.1

Type RM Length L Ch R = 1,6000,455,455,455
BEGIN DESCRIPTION:
Bee Caves Creek 13.0
END DESCRIPTION:
XS GIS Cut Line= 3
      1821475.01     13930524.96      1821525.00     13930375.00
      1821925.02     13930024.99
#Sta/Elev= 30
  4837.5 1972.79  4869.1 1968.98  4900.7 1963.50  4921.8 1934.08  4935.5 1932.51
  4974.5 1932.42  4992.9 1929.93  5010.6 1928.94  5011.1 1928.44  5023.2 1928.94
  5052.0 1930.58  5059.6 1929.93  5115.6 1934.91  5137.5 1935.62  5144.1 1937.37
  5151.7 1937.41  5172.6 1939.59  5180.2 1939.40  5221.9 1942.57  5236.2 1943.35
  5272.2 1943.38  5321.6 1951.13  5328.2 1953.61  5335.8 1954.66  5342.5 1956.65
  5364.3 1960.01  5384.9 1964.54  5448.8 1974.85  5491.5 1980.33  5527.1 1983.14
#Mann=5,-1,0
  4837.5     0.1       0  4935.5    0.07       0  5010.6    0.05       0
  5023.2    0.07       0  5384.9     0.1       0
Bank Sta=5010.6,5023.2
Exp/Cntr=0.3,0.1

Type RM Length L Ch R = 1,5545,470,470,470
BEGIN DESCRIPTION:
Bee Caves Creek 12.0
END DESCRIPTION:
XS GIS Cut Line= 3
      1821675.01     13930724.99      1821925.00     13930525.00
      1822274.97     13930375.01
#Sta/Elev= 30
  4674.1 1966.23  4686.9 1965.34  4730.9 1959.12  4766.1 1951.65  4794.9 1948.83
  4809.4 1945.45  4873.4 1939.55  4894.2 1936.63  4916.6 1936.27  4930.7 1935.03
  4966.2 1930.38  4989.5 1925.29  5064.1 1924.57  5064.6 1924.07  5076.8 1924.57
  5124.8 1925.27  5132.1 1926.10  5137.5 1928.51  5155.6 1929.54  5161.1 1930.74
  5179.5 1931.51  5190.1 1932.68  5255.4 1934.41  5277.1 1936.96  5298.9 1946.94
  5320.6 1961.74  5331.5 1968.03  5342.4 1986.06  5360.5 1989.54  5375.0 1990.41
#Mann=7,-1,0
  4674.1     0.1       0  4686.9    0.07       0  4930.7   0.035       0
  4989.5    0.07       0  5064.1    0.05       0  5076.8    0.07       0
  5179.5     0.1       0
Bank Sta=5064.1,5076.8
Exp/Cntr=0.3,0.1
