--- Contrary Creek.prj (project) ---

Proj Title=Contrary Creek Base Level Engineering
Current Plan=p01
Default Exp/Contr=0.3,0.1
English Units
Geom File=g01
Flow File=f01
Plan File=p01
Y Axis Title=Elevation
X Axis Title(PF)=Main Channel Distance
X Axis Title(XS)=Station
BEGIN DESCRIPTION:
Contrary Creek
END DESCRIPTION:
DSS Export Rating Curves= 0
DSS Export Rating Curve Sorted= 0
DSS Export Volume Flow Curves= 0
DXF OffsetX= 0
DXF OffsetY= 0
DXF ScaleX= 1
DXF ScaleY= 10

--- Contrary Creek.p01 (plan) ---

Plan Title=Multiple Run
Short Identifier=Multiple
Geom File=g01
Flow File=f01
Subcritical Flow
K Sum by GR= 0
Std Step Tol= 0.01
Critical Tol= 0.01
Num of Std Step Trials= 20
Max Error Tol= 0.3
Flow Tol Ratio= 0.001
Split Flow NTrial= 30
Split Flow Tol= 0.02
Split Flow Ratio= 0.02
Log Output Level= 0
Friction Slope Method= 1
Unsteady Friction Slope Method= 2
Unsteady Bridges Friction Slope Method= 1
Parabolic Critical Depth
Global Vel Dist=  1 , 1 , 1
Global Log Level= 0
CheckData=True
Encroach Param= -1, 0, 0, 0
BEGIN DESCRIPTION:
Multiple Run
END DESCRIPTION:

--- Contrary Creek.f01 (steady flow) ---

Flow Title=Multiple
Number of Profiles=7
Profile Names=10-year,25-year,50-year,1pct_min,100-year,1pct_plu,500-year
River Rch & RM= Contrary Creek,Reach-1,35827
     334     524     690     441     880    1755    1408
River Rch & RM= Contrary Creek,Reach-1,34002
    1075    1823    2529    1694    3380    6743    5967
River Rch & RM= Contrary Creek,Reach-1,30001
    1609    2787    3920    2658    5303   10582    9602
River Rch & RM= Contrary Creek,Reach-1,24914
    2180    3837    5454    3734    7450   14864   13755
River Rch & RM= Contrary Creek,Reach-1,24488
    2775    4946    7092    4893    9763   19480   18316
River Rch & RM= Contrary Creek,Reach-1,23178
    2878    5123    7340    5058   10092   20136   18887
River Rch & RM= Contrary Creek,Reach-1,18589
    3356    6013    8652    5985   11942   23827   22523
River Rch & RM= Contrary Creek,Reach-1,15911
    3593    6453    9299    6442   12853   25645   24307
River Rch & RM= Contrary Creek,Reach-1,12168
    4771    8679   12616    8810   17578   35072   33782
River Rch & RM= Contrary Creek,Reach-1,9276
    5042    9191   13379    9354   18664   37240   35961
River Rch & RM= Contrary Creek,Reach-1,8957
    5465    9990   14568   10202   20355   40614   39342
River Rch & RM= Contrary Creek,Reach-1,4486
    5613   10263   14971   10485   20921   41743   40449
Boundary for River Rch & Prof#=Contrary Creek,Reach-1,1
Up Type=0
Dn Type=3
Dn Slope=0.005
Boundary for River Rch & Prof#=Contrary Creek,Reach-1,2
Up Type=0
Dn Type=3
Dn Slope=0.005
Boundary for River Rch & Prof#=Contrary Creek,Reach-1,3
Up Type=0
Dn Type=3
Dn Slope=0.005
Boundary for River Rch & Prof#=Contrary Creek,Reach-1,4
Up Type=0
Dn Type=3
Dn Slope=0.005
Boundary for River Rch & Prof#=Contrary Creek,Reach-1,5
Up Type=0
Dn Type=3
Dn Slope=0.005
Boundary for River Rch & Prof#=Contrary Creek,Reach-1,6
Up Type=0
Dn Type=3
Dn Slope=0.005
Boundary for River Rch & Prof#=Contrary Creek,Reach-1,7
Up Type=0
Dn Type=3
Dn Slope=0.005

--- Contrary Creek.g01 (geometry) ---

Geom Title=Existing Conditions

River Reach=Contrary Creek,Reach-1
Reach XY= 30
      1823375.00     13963075.00      1823350.97     13963302.35
      1824133.30     13963821.93      1825400.09     13963925.21
      1826740.27     13963575.38      1827219.14     13963672.95
      1827572.70     13963280.09      1828530.93     13962927.24
      1829869.14     13962827.07      1830833.15     13963971.63
      1831923.50     13963928.61      1832826.55     13964571.25
      1835077.55     13965480.73      1835568.94     13966066.86
      1836135.17     13966235.33      1836374.62     13966940.27
      1836380.73     13968377.55      1837768.27     13969115.85
      1838519.06     13969027.25      1840050.08     13969775.20
      1841525.00     13969025.00      1842914.50     13968926.22
      1843411.63     13969261.68      1843826.50     13969971.38
      1847145.03     13970724.94      1847923.50     13970571.39
      1849026.55     13969828.75      1849478.65     13969832.73
      1850030.54     13971277.42      1850825.00     13972025.00

Type RM Length L Ch R = 1,35827,445,445,445
BEGIN DESCRIPTION:
Contrary Creek 75.0
END DESCRIPTION:
XS GIS Cut Line= 3
      1823275.02     13963574.98      1823575.00     13963325.00
      1823575.00     13963124.98
#Sta/Elev= 30
  4614.0 2205.62  4635.4 2205.00  4656.3 2203.87  4664.1 2204.11  4678.4 2202.82
  4692.1 2202.28  4705.7 2202.35  4734.4 2200.95  4742.2 2199.72  4748.7 2199.59
  4756.5 2198.76  4791.7 2197.09  4841.1 2196.35  4869.8 2195.29  4876.3 2195.46
  4912.7 2193.55  4976.5 2192.24  4983.0 2192.54  4990.8 2192.28  4995.3 2191.71
  4995.6 2191.21  4999.1 2191.21  4999.3 2191.71  5001.2 2192.59  5007.0 2192.59
  5014.5 2193.91  5034.5 2196.04  5064.5 2197.12  5174.5 2205.61  5204.5 2207.03
#Mann=3,-1,0
  4614.0    0.07       0  4995.3    0.05       0  4999.3    0.07       0
Bank Sta=4995.3,4999.3
Exp/Cntr=0.3,0.1

Type RM Length L Ch R = 1,35382,472,472,472
BEGIN DESCRIPTION:
Contrary Creek 74.0
END DESCRIPTION:
XS GIS Cut Line= 3
      1823675.03     13963824.97      1823925.00     13963575.00
      1823925.00     13963275.01
#Sta/Elev= 30
  4651.3 2196.25  4679.5 2195.51  4693.7 2194.31  4736.1 2193.03  4764.4 2191.75
  4792.7 2190.09  4821.0 2188.92  4863.4 2187.59  4905.8 2186.90  4948.2 2186.58
  4962.4 2186.10  5007.3 2185.18  5014.8 2184.80  5022.8 2184.76  5023.1 2184.26
  5026.6 2184.26  5026.8 2184.76  5034.8 2185.27  5044.8 2185.59  5064.8 2187.29
  5074.8 2187.66  5094.8 2188.81  5104.8 2188.94  5134.8 2189.97  5184.8 2191.29
  5264.8 2196.03  5274.8 2196.24  5294.8 2197.62  5302.3 2198.34  5304.8 2198.34
#Mann=3,-1,0
  4651.3    0.07       0  5022.8    0.05       0  5026.8    0.07       0
Bank Sta=5022.8,5026.8
Exp/Cntr=0.3,0.1

Type RM Length L Ch R = 1,34910,455,455,455
BEGIN DESCRIPTION:
Contrary Creek 73.0
END DESCRIPTION:
XS GIS Cut Line= 3
      1823974.98     13964025.01      1824275.00     13963825.00
      1824225.00     13963224.96
#Sta/Elev= 30
  4639.1 2189.18  4760.8 2184.97  4832.9 2182.98  4863.0 2181.75  4905.0 2181.23
  4914.0 2180.91  4935.1 2179.44  4971.1 2178.60  4977.1 2178.82  4984.2 2178.45
  4984.4 2177.95  4987.9 2177.95  4988.2 2178.45  5009.7 2178.62  5029.8 2179.36
  5039.8 2179.41  5110.1 2181.95  5177.8 2183.31  5190.3 2184.00  5240.5 2184.89
  5280.6 2186.32  5320.8 2186.78  5330.8 2187.25  5391.0 2188.36  5418.6 2190.11
  5441.2 2190.33  5471.3 2191.80  5531.5 2196.97  5551.6 2197.50  5601.8 2200.41
#Mann=3,-1,0
  4639.1    0.07       0  4984.2    0.05       0  4988.2    0.07       0
Bank Sta=4984.2,4988.2
Exp/Cntr=0.3,0.1

Type RM Length L Ch R = 1,34455,453,453,453
BEGIN DESCRIPTION:
Contrary Creek 72.0
END DESCRIPTION:
XS GIS Cut Line= 3
      1824524.98     13964125.04      1824675.00     13963825.00
      1824574.98     13963624.97
#Sta/Elev= 30
  4668.6 2181.22  4691.0 2181.18  4699.4 2180.58  4721.8 2180.11  4727.3 2179.57
  4744.1 2179.31  4758.1 2178.56  4772.1 2178.40  4780.5 2177.80  4839.1 2176.20
  4847.5 2176.36  4883.9 2173.77  4923.0 2171.60  4967.7 2171.82  4981.7 2171.44
  4990.1 2169.95  4993.7 2169.88  4993.9 2169.38  4997.4 2169.38  4997.7 2169.88
  5001.3 2171.04  5006.9 2171.04  5012.4 2171.76  5057.2 2173.67  5062.8 2174.23
  5071.1 2173.95  5129.8 2176.31  5152.2 2177.64  5191.3 2180.72  5227.7 2182.78
#Mann=3,-1,0
  4668.6    0.07       0  4993.7    0.05       0  4997.7    0.07       0
Bank Sta=4993.7,4997.7
Exp/Cntr=0.3,0.1

Type RM Length L Ch R = 1,34002,436,436,436
BEGIN DESCRIPTION:
Contrary Creek 71.0
END DESCRIPTION:
XS GIS Cut Line= 3
      1824924.99     13964125.02      1825075.00     13963875.00
      1825025.01     13963625.03
#Sta/Elev= 30
  4708.4 2175.88  4716.2 2176.01  4722.0 2175.61  4731.8 2175.55  4759.0 2173.82
  4790.1 2173.25  4825.0 2171.96  4832.8 2171.41  4838.7 2172.04  4848.4 2171.71
  4860.0 2170.22  4897.0 2169.06  4928.1 2166.66  4955.3 2165.23  4976.7 2165.15
  4986.4 2165.53  4992.2 2164.98  5030.6 2165.21  5059.2 2164.73  5059.4 2164.23
  5062.9 2164.23  5063.2 2164.73  5071.4 2165.10  5081.6 2166.59  5102.0 2168.57
  5142.7 2171.57  5173.3 2172.71  5203.9 2174.55  5224.3 2174.67  5254.9 2175.56
#Mann=3,-1,0
  4708.4    0.07       0  5059.2    0.05       0  5063.2    0.07       0
Bank Sta=5059.2,5063.2
Exp/Cntr=0.3,0.1

Type RM Length L Ch R = 1,33566,446,446,446
BEGIN DESCRIPTION:
Contrary Creek 70.0
END DESCRIPTION:
XS GIS Cut Line= 3
      1825624.98     13964174.96      1825475.00     13963875.00
      1825324.99     13963574.98
#Sta/Elev= 30
  4669.2 2169.56  4691.5 2168.61  4705.5 2168.51  4722.3 2167.02  4758.6 2166.61
  4781.0 2165.72  4794.9 2164.32  4811.7 2163.53  4817.3 2162.63  4834.1 2161.11
  4856.4 2160.45  4870.4 2160.74  4901.2 2160.13  4927.1 2158.65  4927.4 2158.15
  4930.9 2158.15  4931.1 2158.65  4951.5 2159.39  4968.2 2159.49  4973.8 2160.14
  4990.6 2159.11  5007.4 2158.99  5026.9 2159.96  5049.3 2160.12  5108.0 2161.60
  5152.7 2163.59  5197.4 2166.33  5219.8 2168.21  5303.6 2172.80  5340.0 2173.82
#Mann=3,-1,0
  4669.2    0.07       0  4927.1    0.05       0  4931.1    0.07       0
Bank Sta=4927.1,4931.1
Exp/Cntr=0.3,0.1

Type RM Length L Ch R = 1,33120,464,464,464
BEGIN DESCRIPTION:
Contrary Creek 69.0
END DESCRIPTION:
XS GIS Cut Line= 3
      1825824.99     13964025.03      1825875.00     13963825.00
      1825625.04     13963625.03
#Sta/Elev= 30
  4794.3 2165.78  4858.8 2162.04  4936.1 2155.55  4941.2 2155.78  4959.3 2154.62
  4977.3 2151.96  4982.5 2152.11  4988.2 2151.15  4988.4 2150.65  4991.9 2150.65
  4992.2 2151.15  4997.9 2153.02  5028.5 2154.45  5036.5 2153.92  5042.9 2154.64
  5091.3 2155.07  5114.9 2155.17  5121.3 2155.96  5128.6 2155.86  5135.8 2154.92
  5142.2 2156.31  5150.2 2155.86  5156.6 2157.35  5164.6 2156.97  5171.0 2157.73
  5199.8 2159.07  5220.6 2161.08  5243.0 2161.55  5292.6 2164.13  5320.6 2164.94
#Mann=4,-1,0
  4794.3    0.07       0  4988.2    0.05       0  4992.2    0.07       0
  5091.3     0.1       0
Bank Sta=4988.2,4992.2
Exp/Cntr=0.3,0.1

Type RM Length L Ch R = 1,32656,436,436,436
BEGIN DESCRIPTION:
Contrary Creek 68.0
END DESCRIPTION:
XS GIS Cut Line= 3
      1826275.00     13963925.00      1826275.00     13963725.00
      1826025.01     13963425.01
#Sta/Elev= 30
  4804.6 2157.73  4834.6 2156.59  4854.6 2155.26  4884.6 2154.65  4904.6 2152.84
  4934.6 2151.29  4964.6 2147.55  4972.6 2147.35  4972.8 2146.85  4976.3 2146.85
  4976.6 2147.35  4984.6 2148.19  5032.6 2149.72  5061.2 2149.57  5069.0 2148.64
  5075.5 2149.31  5089.9 2148.83  5118.5 2150.93  5125.0 2151.01  5139.3 2152.82
  5231.7 2156.10  5252.6 2156.44  5274.7 2157.75  5281.2 2157.68  5289.0 2158.70
  5309.8 2158.42  5330.7 2159.08  5373.6 2161.46  5388.0 2162.69  5395.1 2162.53
#Mann=3,-1,0
  4804.6    0.07       0  4972.6    0.05       0  4976.6    0.07       0
Bank Sta=4972.6,4976.6
Exp/Cntr=0.3,0.1

Type RM Length L Ch R = 1,32220,356,356,356
BEGIN DESCRIPTION:
Contrary Creek 67.0
END DESCRIPTION:
XS GIS Cut Line= 3
      1826625.01     13963874.96      1826675.00     13963625.00
      1826525.01     13963425.01
#Sta/Elev= 30
  4740.7 2153.89  4761.1 2152.38  4781.5 2152.03  4842.6 2147.89  4924.2 2144.75
  4965.0 2144.46  4985.4 2143.60  4993.1 2142.89  4998.7 2142.89  5002.9 2142.06
  5015.5 2141.58  5015.7 2141.08  5019.2 2141.08  5019.5 2141.58  5023.7 2141.78
  5032.1 2143.02  5045.6 2143.81  5052.9 2144.85  5088.3 2146.29  5095.6 2147.04
  5109.2 2147.73  5132.1 2148.11  5159.2 2149.63  5188.3 2150.70  5195.6 2151.64
  5209.2 2152.00  5217.5 2152.88  5223.7 2152.68  5232.1 2153.42  5245.6 2153.94
#Mann=3,-1,0
  4740.7    0.07       0  5015.5    0.05       0  5019.5    0.07       0
Bank Sta=5015.5,5019.5
Exp/Cntr=0.3,0.1

Type RM Length L Ch R = 1,31864,526,526,526
BEGIN DESCRIPTION:
Contrary Creek 66.0
END DESCRIPTION:
XS GIS Cut Line= 3
      1826975.00     13963925.04      1827006.34     13963638.64
      1826825.00     13963374.99
#Sta/Elev= 30
  4695.0 2148.77  4725.2 2148.07  4740.7 2147.06  4795.6 2145.63  4825.8 2144.44
  4831.9 2143.94  4896.2 2142.05  4923.1 2140.59  4928.1 2140.92  4936.5 2139.51
  4946.5 2138.87  4956.6 2139.19  4998.0 2138.26  4998.3 2137.76  5001.8 2137.76
  5002.0 2138.26  5008.8 2139.37  5014.9 2139.07  5029.8 2140.05  5036.1 2140.97
  5044.7 2140.94  5050.8 2140.36  5072.5 2140.52  5095.4 2141.69  5122.5 2142.23
  5145.3 2143.81  5188.1 2145.84  5230.3 2146.95  5274.7 2148.97  5303.1 2149.76
#Mann=3,-1,0
  4695.0    0.07       0  4998.0    0.05       0  5002.0    0.07       0
Bank Sta=4998,5002
Exp/Cntr=0.3,0.1

Type RM Length L Ch R = 1,31338,421,421,421
BEGIN DESCRIPTION:
Contrary Creek 65.0
END DESCRIPTION:
XS GIS Cut Line= 3
      1827475.00     13963674.98      1827425.00     13963475.00
      1827175.03     13963175.04
#Sta/Elev= 30
  4788.8 2144.88  4830.0 2143.10  4848.1 2141.49  4853.2 2141.48  4860.9 2140.61
  4902.2 2138.79  4943.4 2135.69  4953.7 2135.77  4984.6 2134.82  4992.4 2134.25
  5002.1 2134.36  5016.4 2135.17  5022.9 2134.38  5030.7 2134.41  5037.2 2133.58
  5043.1 2133.49  5043.3 2132.99  5046.8 2132.99  5047.1 2133.49  5051.6 2134.07
  5065.9 2134.46  5123.2 2137.53  5137.5 2137.76  5172.6 2139.74  5201.3 2140.46
  5236.4 2142.09  5271.5 2142.92  5307.3 2144.97  5321.0 2145.18  5385.4 2149.35
#Mann=3,-1,0
  4788.8    0.07       0  5043.1    0.05       0  5047.1    0.07       0
Bank Sta=5043.1,5047.1
Exp/Cntr=0.3,0.1

Type RM Length L Ch R = 1,30917,439,439,439
BEGIN DESCRIPTION:
Contrary Creek 64.0
END DESCRIPTION:
XS GIS Cut Line= 3
      1827775.00     13963625.02      1827725.00     13963325.00
      1827425.01     13963025.01
#Sta/Elev= 30
  4696.7 2144.10  4737.3 2142.87  4777.8 2140.21  4790.5 2140.03  4828.5 2137.77
  4858.9 2137.52  4869.1 2136.38  4899.5 2135.28  4929.9 2133.17  4980.6 2130.82
  4990.7 2130.97  4996.3 2129.83  4996.6 2129.33  5000.1 2129.33  5000.3 2129.83
  5004.4 2129.83  5015.0 2131.05  5043.3 2132.21  5085.7 2131.59  5099.9 2130.62
  5128.1 2131.11  5170.6 2133.49  5184.7 2133.72  5213.0 2135.80  5227.1 2136.18
  5269.6 2139.38  5326.1 2140.95  5368.6 2143.81  5382.7 2143.97  5425.1 2146.29
#Mann=3,-1,0
  4696.7    0.07       0  4996.3    0.05       0  5000.3    0.07       0
Bank Sta=4996.3,5000.3
Exp/Cntr=0.3,0.1

Type RM Length L Ch R = 1,30478,477,477,477
BEGIN DESCRIPTION:
Contrary Creek 63.0
END DESCRIPTION:
XS GIS Cut Line= 3
      1827974.99     13963475.02      1828075.00     13963175.00
      1827774.97     13962924.98
#Sta/Elev= 30
  4683.8 2136.87  4747.1 2134.43  4768.2 2134.14  4789.2 2132.70  4810.3 2132.50
  4841.9 2130.96  4852.5 2131.22  4863.0 2130.78  4873.6 2129.58  4957.9 2127.07
  4977.0 2124.58  4977.2 2124.08  4980.7 2124.08  4981.0 2124.58  4989.5 2124.80
  4997.4 2125.95  5021.5 2126.58  5042.4 2128.02  5064.5 2127.92  5078.2 2126.45
  5091.8 2125.75  5120.5 2128.08  5142.6 2128.48  5156.3 2129.82  5192.1 2131.46
  5276.7 2134.23  5340.4 2135.52  5369.1 2136.68  5376.9 2137.61  5390.6 2137.44
#Mann=3,-1,0
  4683.8    0.07       0  4977.0    0.05       0  4981.0    0.07       0
Bank Sta=4977,4981
Exp/Cntr=0.3,0.1

Type RM Length L Ch R = 1,30001,466,466,466
BEGIN DESCRIPTION:
Contrary Creek 62.0
END DESCRIPTION:
XS GIS Cut Line= 3
      1828425.00     13963375.03      1828475.00     13962975.00
      1828425.00     13962674.98
#Sta/Elev= 30
  4592.1 2132.01  4629.9 2129.86  4682.8 2128.78  4710.5 2127.31  4715.6 2127.96
  4783.6 2124.79  4823.9 2124.31  4854.2 2122.38  4876.8 2122.40  4914.6 2120.17
  4952.4 2120.79  4997.8 2117.08  5003.3 2115.67  5003.6 2115.17  5007.4 2115.67
  5023.1 2116.71  5028.2 2117.98  5035.8 2117.01  5056.1 2117.04  5083.9 2120.94
  5089.0 2120.55  5096.6 2121.93  5127.0 2124.58  5167.6 2125.61  5198.0 2128.15
  5210.7 2128.11  5258.8 2130.54  5266.4 2131.71  5271.5 2131.38  5299.4 2132.77
#Mann=3,-1,0
  4592.1    0.07       0  5003.3    0.05       0  5007.4    0.07       0
Bank Sta=5003.3,5007.4
Exp/Cntr=0.3,0.1

Type RM Length L Ch R = 1,29535,449,449,449
BEGIN DESCRIPTION:
Contrary Creek 61.0
END DESCRIPTION:
XS GIS Cut Line= 3
      1828974.99     13963224.96      1828925.00     13962925.00
      1828775.02     13962675.04
#Sta/Elev= 30
  4696.0 2126.14  4716.2 2125.83  4723.8 2125.11  4784.7 2122.89  4807.5 2122.94
  4868.3 2121.68  4911.4 2118.64  4919.0 2117.59  4949.4 2116.10  4959.5 2114.72
  4967.1 2112.95  4972.2 2112.85  4979.8 2111.05  4990.0 2110.93  4995.5 2109.18
  4995.8 2108.68  4999.4 2108.68  4999.6 2109.18  5023.4 2109.96  5066.2 2115.34
  5081.7 2115.82  5093.4 2117.26  5116.7 2117.87  5161.4 2121.83  5167.2 2121.53
  5210.0 2122.96  5246.9 2125.48  5268.3 2128.55  5278.0 2128.98  5291.6 2128.56
#Mann=3,-1,0
  4696.0    0.07       0  4995.5    0.05       0  4999.6    0.07       0
Bank Sta=4995.5,4999.6
Exp/Cntr=0.3,0.1

Type RM Length L Ch R = 1,29086,466,466,466
BEGIN DESCRIPTION:
Contrary Creek 60.0
END DESCRIPTION:
XS GIS Cut Line= 3
      1829274.99     13963225.04      1829325.00     13962875.00
      1829075.01     13962575.01
#Sta/Elev= 30
  4646.5 2124.00  4757.7 2118.69  4868.8 2114.47  4909.2 2113.95  4939.5 2112.52
  4990.0 2109.33  4997.6 2107.91  5003.4 2107.91  5005.2 2106.17  5005.5 2105.67
  5009.1 2105.67  5009.4 2106.17  5050.2 2107.58  5085.4 2107.75  5106.2 2109.29
  5114.0 2110.68  5120.5 2110.42  5134.8 2112.38  5149.1 2112.87  5156.3 2113.87
  5177.8 2115.17  5184.3 2116.25  5192.1 2115.92  5206.4 2117.00  5212.9 2116.71
  5255.9 2118.47  5284.5 2118.80  5312.5 2120.39  5348.3 2123.64  5390.6 2124.80
#Mann=3,-1,0
  4646.5    0.07       0  5005.2    0.05       0  5009.4    0.07       0
Bank Sta=5005.2,5009.4
Exp/Cntr=0.3,0.1

Type RM Length L Ch R = 1,28620,477,477,477
BEGIN DESCRIPTION:
Contrary Creek 59.0
END DESCRIPTION:
XS GIS Cut Line= 3
      1829625.00     13963174.99      1829775.00     13962825.00
      1830175.01     13962474.99
#Sta/Elev= 30
  4619.1 2116.20  4680.7 2114.51  4704.3 2114.53  4738.8 2112.61  4785.9 2111.69
  4814.9 2109.44  4869.3 2107.12  4945.5 2105.56  4978.1 2102.10  5007.0 2101.81
  5013.6 2100.25  5021.2 2099.62  5027.9 2100.90  5032.8 2099.58  5033.2 2099.08
  5038.1 2099.58  5042.1 2100.59  5049.7 2100.38  5078.2 2102.79  5084.8 2104.27
  5106.2 2105.32  5248.1 2106.91  5279.3 2108.75  5325.9 2113.01  5340.1 2115.20
  5368.6 2116.92  5382.8 2118.62  5418.0 2120.09  5503.4 2128.72  5531.4 2129.88
#Mann=4,-1,0
  4619.1    0.07       0  5032.8    0.05       0  5038.1    0.07       0
  5279.3     0.1       0
Bank Sta=5032.8,5038.1
Exp/Cntr=0.3,0.1

Type RM Length L Ch R = 1,28143,473,473,473
BEGIN DESCRIPTION:
Contrary Creek 58.0
END DESCRIPTION:
XS GIS Cut Line= 3
      1829924.99     13963225.01      1830175.00     13963025.00
      1830325.02     13962674.96
#Sta/Elev= 30
  4683.9 2111.54  4719.9 2110.41  4769.6 2107.07  4868.8 2103.41  4912.0 2100.42
  4953.6 2098.90  4968.0 2099.27  4987.8 2094.92  4988.2 2094.42  4992.7 2094.42
  4993.2 2094.92  4996.9 2095.60  5000.9 2098.36  5006.8 2098.36  5018.6 2100.40
  5058.5 2098.62  5065.7 2100.08  5094.7 2102.07  5134.6 2102.00  5156.4 2102.84
  5170.9 2104.67  5189.0 2108.05  5210.8 2113.37  5223.5 2115.29  5265.2 2118.74
  5294.0 2122.04  5330.5 2124.94  5370.3 2129.72  5375.8 2129.56  5384.9 2130.44
#Mann=4,-1,0
  4683.9    0.07       0  4987.8    0.05       0  4993.2    0.07       0
  5294.0     0.1       0
Bank Sta=4987.8,4993.2
Exp/Cntr=0.3,0.1

Type RM Length L Ch R = 1,27670,444,444,444
BEGIN DESCRIPTION:
Contrary Creek 57.0
END DESCRIPTION:
XS GIS Cut Line= 3
      1830275.01     13963824.95      1830375.00     13963425.00
      1830774.97     13963025.03
#Sta/Elev= 30
  4588.0 2112.04  4611.1 2111.46  4701.3 2106.28  4804.4 2103.43  4858.5 2100.06
  4899.8 2098.39  4969.3 2096.99  4982.2 2094.52  4990.0 2094.14  4997.7 2095.92
  5003.8 2095.92  5025.8 2093.99  5026.2 2093.49  5031.3 2093.99  5056.8 2096.49
  5085.1 2097.17  5099.3 2096.73  5113.4 2094.19  5127.5 2095.25  5155.8 2095.49
  5170.0 2097.19  5198.3 2096.10  5269.0 2098.74  5325.5 2103.46  5339.7 2103.76
  5368.0 2107.23  5410.4 2114.76  5438.7 2117.59  5509.4 2121.97  5565.9 2127.16
#Mann=3,-1,0
  4588.0    0.07       0  5025.8    0.05       0  5031.3    0.07       0
Bank Sta=5025.8,5031.3
Exp/Cntr=0.3,0.1

Type RM Length L Ch R = 1,27226,419,419,419
BEGIN DESCRIPTION:
Contrary Creek 56.0
END DESCRIPTION:
XS GIS Cut Line= 3
      1830474.99     13964125.02      1830675.00     13963725.00
      1831074.98     13963325.02
#Sta/Elev= 30
  4553.0 2123.15  4583.8 2121.99  4634.1 2116.76  4695.6 2113.37  4740.3 2108.34
  4799.0 2105.75  4835.3 2102.69  4866.1 2101.42  4874.5 2099.41  4880.1 2096.14
  4888.4 2094.14  4910.8 2091.91  4941.5 2093.26  4963.9 2092.07  4977.9 2090.57
  5011.6 2090.02  5012.0 2089.52  5016.7 2089.52  5017.2 2090.02  5042.7 2092.86
  5071.0 2092.61  5099.2 2093.45  5169.9 2092.29  5184.1 2093.85  5240.7 2095.87
  5268.9 2098.07  5353.8 2102.37  5466.9 2112.43  5509.4 2114.46  5565.9 2118.40
#Mann=3,-1,0
  4553.0    0.07       0  5011.6    0.05       0  5017.2    0.07       0
Bank Sta=5011.6,5017.2
Exp/Cntr=0.3,0.1

Type RM Length L Ch R = 1,26807,486,486,486
BEGIN DESCRIPTION:
Contrary Creek 55.0
END DESCRIPTION:
XS GIS Cut Line= 3
      1830825.01     13964124.99      1830925.00     13964025.00
      1831224.99     13963425.02
#Sta/Elev= 30
  4854.6 2106.85  4882.9 2105.21  4967.7 2094.66  4981.9 2090.46  4989.7 2086.52
  4990.1 2086.02  4994.8 2086.02  4995.3 2086.52  5004.4 2086.65  5010.0 2088.27
  5032.3 2088.43  5049.1 2089.30  5077.1 2088.14  5160.9 2090.46  5197.2 2090.80
  5211.2 2090.18  5272.7 2090.80  5300.7 2090.34  5398.5 2092.00  5406.9 2092.85
  5412.5 2092.78  5420.9 2094.78  5434.8 2095.81  5443.2 2097.92  5465.6 2101.22
  5555.0 2108.68  5569.0 2110.76  5583.0 2112.02  5608.1 2115.81  5666.8 2118.11
#Mann=3,-1,0
  4854.6    0.07       0  4989.7    0.05       0  4995.3    0.07       0
Bank Sta=4989.7,4995.3
Exp/Cntr=0.3,0.1

Type RM Length L Ch R = 1,26321,480,480,480
BEGIN DESCRIPTION:
Contrary Creek 54.0
END DESCRIPTION:
XS GIS Cut Line= 3
      1831125.00     13964325.00      1831375.00     13963925.00
      1831525.00     13963574.99
#Sta/Elev= 30
  4528.3 2104.29  4557.2 2102.98  4666.9 2092.81  4717.0 2090.84  4803.7 2089.52
  4834.3 2086.16  4840.2 2086.57  4846.7 2085.15  4861.4 2085.31  4876.8 2086.87
  4928.7 2084.59  4934.6 2085.85  4949.9 2083.15  4964.6 2083.28  4974.2 2082.21
  4974.6 2081.71  4979.9 2082.21  4986.4 2083.90  4992.3 2083.09  4997.1 2084.40
  5032.6 2086.71  5090.7 2087.28  5143.3 2086.47  5161.4 2088.05  5166.8 2087.71
  5195.8 2094.85  5228.5 2101.05  5295.6 2106.78  5348.2 2113.29  5380.8 2115.39
#Mann=3,-1,0
  4528.3    0.07       0  4974.2    0.05       0  4979.9    0.07       0
Bank Sta=4974.2,4979.9
Exp/Cntr=0.3,0.1

Type RM Length L Ch R = 1,25841,456,456,456
BEGIN DESCRIPTION:
Contrary Creek 53.0
END DESCRIPTION:
XS GIS Cut Line= 3
      1831025.00     13964625.00      1831825.00     13963925.00
      1831725.01     13963525.02
#Sta/Elev= 30
  3931.5 2123.14  3967.1 2122.66  4016.4 2119.23  4059.2 2115.34  4087.6 2111.60
  4151.2 2106.81  4292.6 2099.64  4328.7 2096.88  4803.3 2084.22  4852.6 2085.16
  4888.2 2084.56  4916.2 2082.02  4938.0 2081.27  4980.8 2083.16  4997.1 2082.33
  5004.8 2080.61  5014.9 2079.89  5015.3 2079.39  5020.6 2079.89  5025.4 2082.25
  5035.7 2083.16  5118.2 2085.06  5159.4 2087.78  5218.7 2097.82  5252.2 2102.15
  5265.1 2102.69  5324.4 2109.80  5347.6 2111.21  5383.6 2116.52  5406.8 2117.51
#Mann=3,-1,0
  3931.5    0.07       0  5014.9    0.05       0  5020.6    0.07       0
Bank Sta=5014.9,5020.6
Exp/Cntr=0.3,0.1

Type RM Length L Ch R = 1,25385,471,471,471
BEGIN DESCRIPTION:
Contrary Creek 52.0
END DESCRIPTION:
XS GIS Cut Line= 3
      1831425.04     13964574.98      1832225.00     13964075.00
      1832075.00     13963624.99
#Sta/Elev= 30
  4061.6 2100.24  4090.4 2099.73  4127.0 2097.73  4155.9 2097.02  4227.2 2093.92
  4352.2 2091.27  4467.8 2089.67  4604.6 2086.95  4787.4 2081.27  4866.4 2080.71
  4924.2 2081.55  4954.8 2081.25  4982.0 2079.73  4997.3 2077.79  5012.6 2076.64
  5013.1 2076.14  5017.9 2076.14  5018.3 2076.64  5036.6 2079.38  5047.1 2080.01
  5194.7 2083.06  5310.6 2084.20  5352.8 2086.37  5363.3 2087.33  5395.0 2091.79
  5405.5 2094.72  5426.6 2098.24  5437.1 2101.66  5468.8 2105.56  5479.3 2106.08
#Mann=3,-1,0
  4061.6    0.07       0  5012.6    0.05       0  5018.3    0.07       0
Bank Sta=5012.6,5018.3
Exp/Cntr=0.3,0.1

Type RM Length L Ch R = 1,24914,426,426,426
BEGIN DESCRIPTION:
Contrary Creek 51.0
END DESCRIPTION:
XS GIS Cut Line= 3
      1832225.00     13965174.99      1832575.00     13964375.00
      1832975.01     13963974.99
#Sta/Elev= 30
  4126.8 2096.91  4203.2 2093.98  4234.8 2093.43  4287.0 2091.05  4641.8 2083.18
  4727.1 2080.20  4770.8 2077.96  4834.3 2077.81  4857.7 2076.32  4859.2 2075.68
  4859.7 2075.18  4866.7 2075.18  4867.2 2075.68  4901.8 2077.57  4962.2 2078.53
  4985.6 2078.17  5014.1 2076.11  5028.3 2076.34  5042.4 2078.02  5070.7 2075.75
  5113.1 2078.53  5198.0 2078.20  5268.7 2080.00  5325.3 2082.57  5353.6 2084.63
  5410.1 2086.97  5466.7 2091.05  5509.1 2095.35  5537.4 2099.29  5565.7 2101.90
#Mann=3,-1,0
  4126.8    0.07       0  4859.2    0.05       0  4867.2    0.07       0
Bank Sta=4859.2,4867.2
Exp/Cntr=0.3,0.1

Type RM Length L Ch R = 1,24488,455,455,455
BEGIN DESCRIPTION:
Contrary Creek 50.0
END DESCRIPTION:
XS GIS Cut Line= 3
      1832524.98     13964875.01      1832925.00     13964575.00
      1833174.99     13964175.02
#Sta/Elev= 30
  4500.0 2084.41  4650.0 2079.05  4892.7 2074.59  4907.3 2074.92  4928.1 2073.51
  4936.5 2073.76  4957.3 2071.95  4986.5 2070.96  4996.9 2069.57  5003.0 2069.57
  5008.6 2068.37  5009.1 2067.87  5018.1 2067.87  5018.6 2068.37  5023.0 2069.25
  5028.9 2068.79  5035.4 2070.63  5044.2 2072.06  5059.0 2073.17  5065.5 2072.69
  5071.4 2073.04  5086.7 2076.08  5102.0 2078.00  5217.6 2079.60  5275.4 2081.69
  5290.7 2081.56  5342.0 2083.15  5390.9 2085.62  5444.3 2091.11  5471.7 2093.55
#Mann=4,-1,0
  4500.0    0.07       0  5008.6    0.05       0  5018.6    0.07       0
  5444.3     0.1       0
Bank Sta=5008.6,5018.6
Exp/Cntr=0.3,0.1

Type RM Length L Ch R = 1,24033,437,437,437
BEGIN DESCRIPTION:
Contrary Creek 49.0
END DESCRIPTION:
XS GIS Cut Line= 3
      1832525.00     13965525.00      1833325.00     13964725.00
      1833325.00     13964024.97
#Sta/Elev= 30
  3868.9 2115.05  3911.3 2112.28  3953.8 2106.19  3980.8 2103.76  4052.7 2096.91
  4222.5 2089.31  4307.3 2083.28  4363.9 2080.84  4830.6 2072.98  4901.3 2071.54
  4929.6 2069.79  4972.0 2071.06  4986.1 2069.61  4991.7 2067.48  4992.2 2066.98
  5001.8 2067.48  5040.3 2070.25  5080.3 2071.12  5110.3 2069.40  5160.3 2071.40
  5170.3 2073.27  5220.3 2075.79  5370.3 2080.41  5420.3 2084.62  5480.3 2087.67
  5540.5 2093.68  5580.3 2098.23  5640.3 2108.22  5674.4 2110.36  5700.3 2111.54
#Mann=6,-1,0
  3868.9   0.035       0  3980.8    0.07       0  4991.7    0.05       0
  5001.8    0.07       0  5540.5     0.1       0  5674.4    0.07       0
Bank Sta=4991.7,5001.8
Exp/Cntr=0.3,0.1

Type RM Length L Ch R = 1,23596,418,418,418
BEGIN DESCRIPTION:
Contrary Creek 48.0
END DESCRIPTION:
XS GIS Cut Line= 3
      1833338.18     13965441.57      1833725.00     13964825.00
      1833874.99     13964575.01
#Sta/Elev= 30
  4267.5 2081.63  4327.9 2080.05  4357.9 2080.05  4364.4 2079.05  4501.1 2075.42
  4547.7 2075.00  4636.9 2073.84  4865.5 2070.83  4900.9 2069.03  4936.3 2065.85
  4951.2 2065.23  4972.4 2062.60  4987.7 2062.39  4992.4 2061.41  5003.1 2061.96
  5003.8 2061.17  5004.3 2060.67  5013.7 2060.67  5014.2 2061.17  5018.7 2061.91
  5040.1 2061.92  5045.9 2063.02  5053.7 2065.67  5067.3 2067.59  5088.7 2069.00
  5156.7 2071.15  5162.5 2070.61  5193.6 2071.59  5263.6 2076.61  5286.9 2077.67
#Mann=5,-1,0
  4267.5    0.07       0  4547.7     0.1       0  4636.9    0.07       0
  5003.8    0.05       0  5014.2    0.07       0
Bank Sta=5003.8,5014.2
Exp/Cntr=0.3,0.1

Type RM Length L Ch R = 1,23178,471,471,471
BEGIN DESCRIPTION:
Contrary Creek 47.0
END DESCRIPTION:
XS GIS Cut Line= 3
      1833700.07     13965452.18      1834075.00     13965025.00
      1834345.76     13964675.10
#Sta/Elev= 30
  4436.3 2076.96  4466.2 2076.67  4480.4 2075.49  4501.3 2074.80  4600.9 2073.15
  4621.8 2072.08  4791.8 2069.53  4834.4 2067.21  4877.0 2065.59  4898.2 2063.69
  4919.7 2063.29  4948.2 2061.13  4969.1 2060.89  4983.3 2057.28  4992.3 2056.28
  4992.8 2055.78  5002.4 2055.78  5002.9 2056.28  5004.7 2057.03  5018.2 2056.75
  5032.7 2062.54  5040.9 2064.13  5061.7 2066.00  5068.0 2065.79  5126.0 2068.26
  5155.0 2068.81  5240.1 2074.50  5354.2 2077.30  5424.8 2083.24  5447.1 2084.08
#Mann=3,-1,0
  4436.3    0.07       0  4992.3    0.05       0  5002.9    0.07       0
Bank Sta=4992.3,5002.9
Exp/Cntr=0.3,0.1

Type RM Length L Ch R = 1,22707,450,450,450
BEGIN DESCRIPTION:
Contrary Creek 46.0
END DESCRIPTION:
XS GIS Cut Line= 3
      1834149.86     13965664.73      1834475.00     13965225.00
      1834629.58     13964919.24
#Sta/Elev= 30
  4453.1 2075.45  4538.3 2073.41  4671.2 2069.91  4721.3 2066.64  4750.6 2067.18
  4800.7 2062.97  4827.9 2062.02  4836.1 2063.38  4840.8 2062.59  4857.0 2062.24
  4863.2 2060.71  4906.7 2060.01  4921.7 2057.24  4936.3 2056.42  4963.4 2056.42
  4978.0 2055.28  4987.3 2052.88  4987.8 2052.38  4998.0 2052.88  5000.0 2054.52
  5008.3 2055.97  5013.9 2055.69  5030.6 2059.40  5036.2 2059.02  5097.5 2069.32
  5119.8 2069.76  5134.4 2071.61  5275.8 2078.29  5336.1 2081.57  5342.6 2082.69
#Mann=6,-1,0
  4453.1     0.1       0  4538.3    0.07       0  4827.9   0.035       0
  4840.8    0.07       0  4987.3    0.05       0  4998.0    0.07       0
Bank Sta=4987.3,4998
Exp/Cntr=0.3,0.1

Type RM Length L Ch R = 1,22257,462,462,462
BEGIN DESCRIPTION:
Contrary Creek 45.0
END DESCRIPTION:
XS GIS Cut Line= 3
      1834403.99     13965988.99      1834875.00     13965375.00
      1834875.00     13965275.04
#Sta/Elev= 30
  4230.9 2078.97  4291.4 2077.87  4312.2 2076.66  4446.6 2073.98  4499.0 2070.65
  4548.8 2062.30  4569.6 2060.62  4605.0 2059.69  4663.0 2059.95  4698.4 2058.89
  4719.2 2057.46  4733.8 2057.53  4762.7 2059.20  4790.5 2058.14  4818.9 2058.99
  4862.4 2061.44  4926.8 2060.72  4947.6 2058.95  4976.7 2051.76  4985.8 2051.42
  4986.3 2050.92  4996.1 2050.92  4996.6 2051.42  5001.6 2053.15  5007.2 2053.15
  5014.7 2058.09  5034.7 2067.58  5044.7 2069.91  5082.4 2071.25  5104.7 2072.14
#Mann=6,-1,0
  4230.9    0.07       0  4446.6   0.035       0  4733.8    0.07       0
  4985.8    0.05       0  4996.6    0.07       0  5082.4     0.1       0
Bank Sta=4985.8,4996.6
Exp/Cntr=0.3,0.1

Type RM Length L Ch R = 1,21795,441,441,441
BEGIN DESCRIPTION:
Contrary Creek 44.0
END DESCRIPTION:
XS GIS Cut Line= 3
      1834874.97     13966025.04      1835225.00     13965625.00
      1835225.00     13965474.95
#Sta/Elev= 30
  4476.5 2073.13  4483.7 2072.53  4504.5 2072.54  4547.3 2068.21  4561.5 2065.41
  4575.7 2061.62  4582.8 2056.49  4590.0 2053.01  4625.1 2053.41  4632.7 2055.02
  4646.9 2056.34  4724.7 2057.83  4845.3 2057.81  4908.9 2057.11  4927.0 2055.92
  4944.0 2051.97  4958.2 2051.56  4965.8 2052.10  4981.3 2047.91  4981.8 2047.41
  4991.6 2047.41  4992.1 2047.91  4994.3 2051.79  5000.9 2054.50  5028.1 2054.57
  5058.1 2056.89  5088.1 2061.17  5108.1 2063.15  5128.1 2066.89  5158.1 2070.25
#Mann=4,-1,0
  4476.5   0.035       0  4927.0    0.07       0  4981.3    0.05       0
  4992.1    0.07       0
Bank Sta=4981.3,4992.1
Exp/Cntr=0.3,0.1

Type RM Length L Ch R = 1,21354,452,452,452
BEGIN DESCRIPTION:
Contrary Creek 43.0
END DESCRIPTION:
XS GIS Cut Line= 3
      1835175.02     13966174.99      1835475.00     13965975.00
      1835874.97     13965725.02
#Sta/Elev= 30
  4639.5 2070.31  4668.0 2070.21  4683.0 2069.36  4698.1 2067.45  4704.1 2065.30
  4725.1 2060.37  4747.6 2056.16  4797.2 2055.10  4878.3 2050.59  4905.4 2052.15
  4920.4 2051.70  4927.9 2050.67  4964.0 2049.99  4981.0 2048.42  4981.5 2047.92
  4992.1 2048.42  4997.0 2049.60  5003.0 2049.60  5013.6 2051.36  5028.3 2052.24
  5094.4 2052.78  5123.3 2054.66  5211.7 2055.73  5272.3 2057.39  5306.0 2058.22
  5327.3 2060.15  5333.2 2061.70  5400.4 2070.36  5442.8 2077.48  5471.7 2077.82
#Mann=5,-1,0
  4639.5   0.035       0  4981.0   0.035       0  4992.1   0.035       0
  5028.3    0.07       0  5272.3     0.1       0
Bank Sta=4981,4992.1
Exp/Cntr=0.3,0.1

Type RM Length L Ch R = 1,20902,454,454,454
BEGIN DESCRIPTION:
Contrary Creek 42.0
END DESCRIPTION:
XS GIS Cut Line= 3
      1835475.01     13966524.99      1835875.00     13966125.00
      1836075.02     13965974.99
#Sta/Elev= 30
  4438.6 2064.50  4481.0 2062.61  4537.6 2058.62  4646.0 2056.11  4763.9 2053.32
  4820.4 2050.32  4862.9 2049.35  4877.0 2048.34  4919.4 2047.97  4947.7 2044.87
  4970.4 2043.75  4970.9 2043.25  4981.6 2043.75  4990.1 2043.94  5000.7 2047.17
  5007.4 2047.17  5032.4 2049.85  5111.6 2049.81  5140.7 2051.88  5147.0 2054.24
  5160.5 2056.64  5167.8 2061.08  5176.2 2063.01  5182.4 2067.62  5190.7 2070.29
  5197.0 2073.22  5217.8 2079.30  5226.2 2080.49  5253.9 2080.87  5254.3 2080.87
#Mann=5,-1,0
  4438.6   0.035       0  4646.0    0.07       0  4970.4    0.05       0
  4981.6    0.07       0  5253.9     0.1       0
Bank Sta=4970.4,4981.6
Exp/Cntr=0.3,0.1

Type RM Length L Ch R = 1,20448,451,451,451
BEGIN DESCRIPTION:
Contrary Creek 41.0
END DESCRIPTION:
XS GIS Cut Line= 3
      1835824.96     13966575.02      1836175.00     13966375.00
      1836275.01     13966274.99
#Sta/Elev= 30
  4592.2 2055.65  4615.3 2055.35  4643.4 2054.42  4657.7 2054.38  4730.5 2053.68
  4776.5 2052.36  4783.0 2051.87  4811.1 2051.62  4842.0 2050.05  4869.4 2049.51
  4906.8 2047.78  4922.7 2046.20  4944.2 2042.64  4950.0 2042.48  4965.8 2043.41
  4981.7 2042.89  4992.5 2041.33  4998.9 2041.33  5003.9 2040.34  5004.4 2039.84
  5014.6 2039.84  5015.1 2040.34  5023.6 2041.38  5037.8 2044.44  5066.1 2062.07
  5094.4 2074.25  5108.5 2079.20  5122.6 2080.58  5133.2 2082.28  5136.8 2082.28
#Mann=4,-1,0
  4592.2   0.035       0  4657.7    0.07       0  5003.9    0.05       0
  5015.1    0.07       0
Bank Sta=5003.9,5015.1
Exp/Cntr=0.3,0.1

Type RM Length L Ch R = 1,19997,481,481,481
BEGIN DESCRIPTION:
Contrary Creek 40.0
END DESCRIPTION:
XS GIS Cut Line= 3
      1835925.01     13966675.00      1836325.00     13966775.00
      1836474.98     13966625.02
#Sta/Elev= 30
  4587.7 2054.12  4628.9 2053.17  4640.4 2053.26  4701.1 2051.94  4793.8 2046.97
  4853.1 2045.39  4858.3 2045.57  4876.3 2043.98  4894.3 2043.03  4907.2 2042.79
  4917.5 2041.29  4935.6 2040.08  4940.7 2039.43  4969.1 2039.62  4976.8 2038.71
  4989.7 2038.77  4991.8 2038.08  4992.3 2037.58  5002.5 2037.58  5003.0 2038.08
  5028.3 2039.47  5042.4 2041.49  5056.6 2045.44  5084.9 2054.15  5099.0 2057.68
  5141.4 2065.58  5169.7 2072.57  5183.8 2075.56  5198.0 2077.45  5212.1 2078.09
#Mann=4,-1,0
  4587.7   0.035       0  4640.4    0.07       0  4991.8    0.05       0
  5003.0    0.07       0
Bank Sta=4991.8,5003
Exp/Cntr=0.3,0.1

Type RM Length L Ch R = 1,19516,479,479,479
BEGIN DESCRIPTION:
Contrary Creek 39.0
END DESCRIPTION:
XS GIS Cut Line= 3
      1835924.99     13967075.00      1836325.00     13967225.00
      1836474.97     13967175.01
#Sta/Elev= 30
  4568.5 2051.72  4621.9 2049.92  4669.1 2049.31  4694.0 2047.74  4778.0 2045.00
  4784.8 2045.09  4809.7 2043.63  4834.6 2042.86  4870.2 2042.51  4888.9 2040.76
  4895.1 2038.54  4900.5 2038.62  4925.4 2036.84  4950.3 2038.35  4974.4 2037.96
  4980.6 2037.03  4998.3 2036.51  5000.6 2035.19  5001.1 2034.69  5011.4 2034.69
  5011.9 2035.19  5027.3 2036.15  5037.9 2035.26  5048.4 2035.83  5059.0 2039.44
  5069.5 2042.27  5101.1 2047.63  5122.2 2050.50  5132.7 2050.56  5153.8 2052.09
#Mann=4,-1,0
  4568.5   0.035       0  4778.0    0.07       0  5000.6    0.05       0
  5011.9    0.07       0
Bank Sta=5000.6,5011.9
Exp/Cntr=0.3,0.1

Type RM Length L Ch R = 1,19037,448,448,448
BEGIN DESCRIPTION:
Contrary Creek 38.0
END DESCRIPTION:
XS GIS Cut Line= 3
      1835310.57     13967483.12      1836325.00     13967675.00
      1836624.96     13967575.01
#Sta/Elev= 30
  3967.5 2077.39  4053.3 2074.90  4073.8 2074.98  4168.2 2071.74  4206.1 2068.69
  4215.5 2068.59  4226.4 2066.20  4307.9 2060.67  4318.0 2060.73  4330.3 2058.98
  4338.4 2059.40  4389.3 2056.36  4419.8 2056.00  4521.6 2051.85  4643.7 2048.32
  4694.6 2045.64  4725.1 2045.77  4735.3 2044.35  4869.0 2037.83  4877.8 2035.50
  4921.4 2035.14  4938.8 2033.47  4973.9 2032.34  4974.4 2031.84  4985.3 2032.34
  5021.0 2033.14  5063.2 2036.84  5126.4 2037.92  5158.0 2041.14  5316.1 2049.95
#Mann=3,-1,0
  3967.5    0.07       0  4973.9    0.05       0  4985.3    0.07       0
Bank Sta=4973.9,4985.3
Exp/Cntr=0.3,0.1

Type RM Length L Ch R = 1,18589,447,447,447
BEGIN DESCRIPTION:
Contrary Creek 37.0
END DESCRIPTION:
XS GIS Cut Line= 3
      1835798.87     13968390.26      1836275.00     13968075.00
      1836825.03     13967724.98
#Sta/Elev= 30
  4429.9 2060.85  4451.9 2059.14  4488.0 2057.64  4713.1 2052.32  4761.7 2050.08
  4770.8 2050.39  4828.0 2047.80  4849.0 2045.86  4879.1 2045.40  4951.3 2037.20
  4987.4 2031.25  4993.4 2031.38  4997.9 2029.50  5000.9 2029.50  5002.2 2027.99
  5002.7 2027.49  5014.5 2027.49  5015.0 2027.99  5045.0 2029.79  5060.2 2028.97
  5087.3 2031.17  5095.8 2030.48  5108.5 2030.78  5123.7 2032.10  5131.3 2033.73
  5138.9 2036.33  5181.3 2039.04  5290.5 2041.26  5426.0 2045.22  5652.9 2052.91
#Mann=4,-1,0
  4429.9    0.07       0  5002.2    0.05       0  5015.0    0.07       0
  5426.0   0.035       0
Bank Sta=5002.2,5015
Exp/Cntr=0.3,0.1

Type RM Length L Ch R = 1,18142,442,442,442
BEGIN DESCRIPTION:
Contrary Creek 36.0
END DESCRIPTION:
XS GIS Cut Line= 3
      1836425.01     13968624.97      1836475.00     13968425.00
      1836824.97     13968175.02
#Sta/Elev= 30
  4798.3 2051.63  4870.4 2049.03  4880.7 2049.00  4891.0 2048.45  4903.9 2047.08
  4932.3 2046.66  4940.0 2044.44  4945.2 2040.73  4952.9 2036.36  4963.2 2029.76
  4974.8 2023.56  4975.3 2023.06  4987.2 2023.06  4987.7 2023.56  5007.5 2023.72
  5011.8 2024.14  5017.9 2026.42  5032.7 2027.42  5062.2 2030.60  5097.8 2031.42
  5118.7 2032.76  5148.2 2033.64  5225.6 2037.25  5234.2 2037.13  5249.0 2038.03
  5290.8 2038.80  5355.9 2041.43  5362.0 2091.26  5370.6 2041.91  5434.5 2044.58
#Mann=3,-1,0
  4798.3    0.07       0  4974.8    0.05       0  4987.7    0.07       0
Bank Sta=4974.8,4987.7
Exp/Cntr=0.3,0.1

Type RM Length L Ch R = 1,17700,430,430,430
BEGIN DESCRIPTION:
Contrary Creek 35.0
END DESCRIPTION:
XS GIS Cut Line= 3
      1836825.00     13968875.03      1836825.00     13968675.00
      1837025.01     13968424.99
#Sta/Elev= 30
  4795.8 2043.24  4805.8 2043.19  4865.8 2039.35  4875.8 2039.37  4905.8 2036.75
  4925.8 2034.43  4965.8 2031.73  4985.8 2029.87  4993.3 2025.02  4999.0 2025.02
  5002.9 2020.19  5003.4 2019.69  5015.5 2019.69  5016.0 2020.19  5038.3 2021.02
  5059.9 2026.46  5067.1 2027.10  5073.5 2026.20  5081.9 2026.01  5095.9 2025.64
  5115.9 2026.35  5123.9 2028.40  5131.1 2029.47  5151.9 2028.78  5166.3 2029.57
  5209.5 2033.64  5223.9 2034.34  5259.2 2038.21  5288.0 2040.72  5316.0 2041.94
#Mann=4,-1,0
  4795.8     0.1       0  5002.9    0.05       0  5016.0     0.1       0
  5081.9    0.07       0
Bank Sta=5002.9,5016
Exp/Cntr=0.3,0.1

Type RM Length L Ch R = 1,17270,443,443,443
BEGIN DESCRIPTION:
Contrary Creek 34.0
END DESCRIPTION:
XS GIS Cut Line= 3
      1837024.98     13969075.04      1837225.00     13968775.00
      1837324.99     13968475.03
#Sta/Elev= 30
  4634.8 2046.60  4663.4 2046.16  4756.5 2039.06  4792.6 2035.03  4801.6 2034.72
  4837.7 2031.14  4843.7 2029.26  4851.2 2028.70  4864.7 2026.36  4900.8 2022.62
  4909.8 2023.74  4930.8 2023.69  4936.8 2024.47  4945.8 2024.24  4951.8 2023.24
  4981.9 2022.40  4985.8 2021.32  4986.3 2020.82  4998.5 2020.82  4999.0 2021.32
  5037.6 2024.95  5048.1 2029.18  5058.6 2031.43  5069.2 2032.18  5079.7 2034.10
  5153.5 2039.00  5164.1 2038.46  5222.8 2040.60  5290.5 2044.86  5311.6 2045.46
#Mann=5,-1,0
  4634.8     0.1       0  4981.9    0.07       0  4985.8    0.05       0
  4999.0    0.07       0  5222.8     0.1       0
Bank Sta=4985.8,4999
Exp/Cntr=0.3,0.1

Type RM Length L Ch R = 1,16827,449,449,449
BEGIN DESCRIPTION:
Contrary Creek 33.0
END DESCRIPTION:
XS GIS Cut Line= 3
      1837525.00     13969224.99      1837575.00     13969025.00
      1837625.00     13968675.00
#Sta/Elev= 30
  4789.5 2038.33  4797.9 2038.13  4841.0 2036.36  4882.3 2032.62  4890.0 2030.63
  4895.1 2030.06  4902.9 2027.52  4913.2 2023.23  4923.5 2020.93  4931.2 2020.17
  4944.1 2020.39  4954.4 2021.68  4964.7 2021.07  4972.5 2021.84  4977.6 2020.42
  4985.3 2019.88  4986.5 2017.90  4987.0 2017.40  4999.2 2017.40  4999.7 2017.90
  5026.0 2018.51  5046.2 2019.85  5056.3 2021.25  5066.4 2023.96  5116.9 2027.42
  5150.0 2030.88  5197.7 2033.71  5238.1 2034.69  5338.3 2039.00  5349.2 2039.56
#Mann=6,-1,0
  4789.5   0.035       0  4797.9    0.07       0  4986.5    0.05       0
  4999.7    0.07       0  5150.0   0.035       0  5338.3    0.07       0
Bank Sta=4986.5,4999.7
Exp/Cntr=0.3,0.1

Type RM Length L Ch R = 1,16378,467,467,467
BEGIN DESCRIPTION:
Contrary Creek 32.0
END DESCRIPTION:
XS GIS Cut Line= 3
      1837699.20     13969501.22      1837975.00     13969075.00
      1838075.01     13968674.98
#Sta/Elev= 30
  4492.3 2041.18  4660.0 2036.75  4675.1 2037.35  4702.2 2035.84  4847.3 2034.66
  4868.9 2033.27  4883.6 2031.34  4892.8 2029.02  4913.9 2017.06  4919.8 2017.97
  4941.0 2015.16  4956.1 2015.15  4970.6 2013.20  4971.1 2012.70  4983.8 2013.20
  4986.4 2014.84  4997.0 2016.08  5023.2 2016.93  5041.2 2018.98  5072.1 2020.36
  5105.6 2020.34  5113.4 2022.34  5185.4 2028.54  5195.8 2028.60  5224.2 2032.00
  5257.7 2033.59  5300.1 2037.25  5340.1 2039.61  5394.2 2045.74  5412.3 2046.79
#Mann=5,-1,0
  4492.3    0.07       0  4970.6    0.05       0  4983.8    0.07       0
  5185.4   0.035       0  5300.1    0.07       0
Bank Sta=4970.6,4983.8
Exp/Cntr=0.3,0.1

Type RM Length L Ch R = 1,15911,447,447,447
BEGIN DESCRIPTION:
Contrary Creek 31.0
END DESCRIPTION:
XS GIS Cut Line= 3
      1838314.09     13969458.97      1838425.00     13969025.00
      1838475.01     13968824.97
#Sta/Elev= 30
  4551.6 2037.13  4619.3 2036.13  4674.6 2033.93  4695.8 2033.27  4701.0 2032.50
  4720.8 2032.38  4736.7 2030.32  4772.3 2028.56  4782.8 2027.08  4803.4 2026.34
  4824.0 2024.02  4859.2 2021.98  4875.7 2017.74  4900.0 2015.74  4927.3 2011.97
  4947.9 2011.39  4968.5 2012.76  4990.0 2010.75  4990.5 2010.25  5003.3 2010.25
  5003.8 2010.75  5017.6 2012.18  5022.7 2011.98  5051.1 2019.74  5058.8 2023.06
  5063.9 2023.64  5082.0 2030.78  5141.2 2039.40  5168.9 2041.77  5205.7 2043.95
#Mann=5,-1,0
  4551.6     0.1       0  4674.6    0.07       0  4990.0    0.05       0
  5003.8    0.07       0  5168.9     0.1       0
Bank Sta=4990,5003.8
Exp/Cntr=0.3,0.1

Type RM Length L Ch R = 1,15464,425,425,425
BEGIN DESCRIPTION:
Contrary Creek 30.0
END DESCRIPTION:
XS GIS Cut Line= 3
      1838632.06     13969675.59      1838825.00     13969175.00
      1838825.00     13968974.99
#Sta/Elev= 30
  4458.9 2040.50  4478.3 2040.39  4517.5 2038.29  4587.5 2035.89  4609.6 2034.40
  4647.4 2029.85  4663.2 2029.63  4695.3 2026.94  4707.4 2026.88  4738.2 2023.24
  4748.9 2023.18  4781.3 2020.52  4802.5 2019.19  4877.5 2017.52  4909.6 2015.80
  4931.2 2011.96  4963.2 2010.85  4974.0 2008.94  4980.4 2006.42  5005.4 2003.75
  5008.5 2001.76  5009.0 2001.26  5022.3 2001.76  5025.4 2003.61  5035.4 2006.41
  5045.4 2017.34  5055.4 2022.26  5105.4 2034.30  5165.4 2039.69  5195.4 2040.40
#Mann=5,-1,0
  4458.9    0.07       0  4517.5     0.1       0  4781.3    0.07       0
  5008.5    0.05       0  5022.3    0.07       0
Bank Sta=5008.5,5022.3
Exp/Cntr=0.3,0.1

Type RM Length L Ch R = 1,15039,424,424,424
BEGIN DESCRIPTION:
Contrary Creek 29.0
END DESCRIPTION:
XS GIS Cut Line= 3
      1839025.01     13969774.98      1839175.00     13969375.00
      1839374.98     13969075.03
#Sta/Elev= 30
  4568.4 2036.43  4613.8 2034.09  4685.9 2027.21  4693.9 2027.41  4699.2 2026.11
  4721.4 2025.26  4803.3 2021.53  4846.1 2016.88  4888.8 2014.05  4919.4 2008.80
  4925.3 2006.58  4931.5 2006.20  4963.5 2007.70  4974.2 2007.34  4980.5 2005.34
  5002.1 2004.60  5002.6 2004.10  5016.1 2004.60  5039.1 2006.02  5060.2 2010.46
  5096.2 2014.86  5103.7 2014.95  5117.3 2017.49  5162.3 2020.37  5204.4 2021.50
  5225.4 2024.87  5276.5 2029.55  5284.0 2031.07  5327.6 2034.86  5356.1 2035.25
#Mann=5,-1,0
  4568.4    0.07       0  4721.4     0.1       0  4919.4    0.07       0
  5002.1    0.05       0  5016.1    0.07       0
Bank Sta=5002.1,5016.1
Exp/Cntr=0.3,0.1

Type RM Length L Ch R = 1,14615,425,425,425
BEGIN DESCRIPTION:
Contrary Creek 28.0
END DESCRIPTION:
XS GIS Cut Line= 3
      1839474.99     13969925.04      1839525.00     13969575.00
      1839624.99     13969275.02
#Sta/Elev= 30
  4646.4 2041.12  4676.7 2038.95  4727.2 2032.78  4747.5 2030.91  4808.1 2023.12
  4848.5 2020.14  4868.7 2016.31  4878.8 2013.09  4888.9 2009.07  4899.0 2004.23
  4909.1 2004.33  4912.1 2003.32  4912.6 2002.82  4925.7 2002.82  4926.2 2003.32
  4949.5 2005.24  4969.7 2006.00  4979.8 2005.06  4989.9 2003.35  5010.5 2004.84
  5063.2 2005.43  5084.3 2010.58  5105.4 2013.53  5147.6 2017.14  5168.6 2017.70
  5179.2 2018.65  5221.3 2020.59  5237.2 2020.87  5284.6 2023.62  5316.2 2024.20
#Mann=3,-1,0
  4646.4    0.07       0  4912.1    0.05       0  4926.2    0.07       0
Bank Sta=4912.1,4926.2
Exp/Cntr=0.3,0.1

Type RM Length L Ch R = 1,14190,483,483,483
BEGIN DESCRIPTION:
Contrary Creek 27.0
END DESCRIPTION:
XS GIS Cut Line= 3
      1839875.00     13969975.03      1839875.00     13969775.00
      1839825.00     13969424.98
#Sta/Elev= 30
  4795.0 2040.93  4835.0 2037.81  4875.0 2032.43  4915.0 2027.96  4935.0 2024.79
  4955.0 2023.28  4965.0 2018.76  4985.0 2003.64  4992.5 1998.58  4997.6 1998.58
  5005.1 1995.95  5008.2 1995.57  5008.7 1995.07  5021.8 1995.07  5022.3 1995.57
  5025.3 1996.06  5035.4 1999.12  5075.8 2003.07  5085.9 2002.32  5096.0 2004.16
  5106.1 2004.60  5126.3 2007.52  5136.4 2008.49  5156.7 2008.51  5207.2 2010.32
  5257.7 2013.58  5267.8 2014.67  5277.9 2014.77  5308.2 2016.67  5348.6 2018.24
#Mann=3,-1,0
  4795.0    0.07       0  5008.2    0.05       0  5022.3    0.07       0
Bank Sta=5008.2,5022.3
Exp/Cntr=0.3,0.1

Type RM Length L Ch R = 1,13707,446,446,446
BEGIN DESCRIPTION:
Contrary Creek 26.0
END DESCRIPTION:
XS GIS Cut Line= 3
      1840375.01     13969875.05      1840325.00     13969675.00
      1840175.00     13969275.00
#Sta/Elev= 30
  4793.8 2023.23  4845.4 2021.42  4858.3 2019.53  4876.3 2019.09  4894.3 2016.74
  4917.5 2012.82  4927.8 2009.19  4935.6 2001.57  4940.7 2000.00  4948.5 1996.09
  4969.1 1996.04  4976.8 1995.44  4982.0 1995.82  4990.3 1994.50  4990.8 1994.00
  5004.0 1994.00  5004.5 1994.50  5009.8 1995.52  5045.4 1997.51  5075.7 2001.49
  5100.6 2005.97  5210.9 2008.05  5266.1 2010.08  5271.5 2010.77  5309.7 2012.35
  5351.6 2015.21  5356.9 2015.06  5363.1 2016.23  5395.2 2019.01  5427.2 2019.91
#Mann=3,-1,0
  4793.8    0.07       0  4990.3    0.05       0  5004.5    0.07       0
Bank Sta=4990.3,5004.5
Exp/Cntr=0.3,0.1

Type RM Length L Ch R = 1,13261,453,453,453
BEGIN DESCRIPTION:
Contrary Creek 25.0
END DESCRIPTION:
XS GIS Cut Line= 3
      1840725.00     13969724.95      1840725.00     13969525.00
      1840456.70     13968935.87
#Sta/Elev= 30
  4795.5 2020.43  4823.5 2019.28  4855.5 2017.15  4885.5 2013.04  4905.5 2011.73
  4925.5 2007.69  4935.5 2004.33  4955.5 2000.02  4965.5 1987.18  4995.5 1985.58
  4997.1 1984.47  4997.6 1983.97  5011.3 1984.47  5017.4 1987.74  5032.8 1990.70
  5039.4 1993.68  5055.8 1995.93  5061.4 1998.13  5130.5 2002.45  5176.6 2003.53
  5205.1 2005.54  5228.2 2005.65  5281.1 2009.11  5320.4 2010.56  5336.1 2012.37
  5348.9 2012.26  5471.9 2019.23  5567.4 2022.18  5617.7 2026.01  5642.8 2027.95
#Mann=6,-1,0
  4795.5   0.035       0  4823.5    0.07       0  4997.1    0.05       0
  5011.3    0.07       0  5471.9     0.1       0  5617.7   0.035       0
Bank Sta=4997.1,5011.3
Exp/Cntr=0.3,0.1

Type RM Length L Ch R = 1,12808,467,467,467
BEGIN DESCRIPTION:
Contrary Creek 24.0
END DESCRIPTION:
XS GIS Cut Line= 3
      1841125.00     13969574.99      1841125.00     13969375.00
      1840925.00     13969025.00
#Sta/Elev= 30
  4796.2 2014.54  4826.2 2013.45  4856.2 2010.67  4876.2 2009.81  4926.2 2005.16
  4956.2 2000.09  4976.2 1998.85  4986.2 1997.29  4993.7 1993.94  4999.1 1993.94
  5004.1 1989.96  5019.2 1985.99  5025.7 1986.63  5040.2 1985.76  5040.7 1985.26
  5054.5 1985.76  5068.9 1987.63  5076.8 1986.68  5090.5 1986.65  5099.8 1987.90
  5106.3 1991.06  5127.9 1995.15  5157.4 1998.12  5208.5 2000.27  5224.4 2001.78
  5238.1 2001.74  5273.3 2005.43  5318.7 2007.39  5370.3 2011.84  5399.3 2013.06
#Mann=4,-1,0
  4796.2    0.07       0  5040.2    0.05       0  5054.5    0.07       0
  5370.3     0.1       0
Bank Sta=5040.2,5054.5
Exp/Cntr=0.3,0.1

Type RM Length L Ch R = 1,12341,173,173,173
BEGIN DESCRIPTION:
Contrary Creek 23.0
END DESCRIPTION:
XS GIS Cut Line= 3
      1841524.99     13969474.96      1841425.00     13969075.00
      1841175.02     13969025.00
#Sta/Elev= 30
  4592.2 2021.59  4656.6 2015.77  4692.7 2010.80  4733.9 2007.39  4739.0 2007.75
  4746.8 2005.91  4775.1 2002.80  4808.6 2000.83  4816.4 1999.51  4862.7 1996.23
  4880.8 1992.17  4891.1 1988.23  4904.0 1985.88  4952.9 1984.73  4986.4 1985.05
  4994.7 1984.39  4995.2 1983.89  5008.5 1983.89  5009.0 1984.39  5014.7 1985.91
  5045.3 1984.91  5075.9 1990.33  5086.1 1994.19  5106.5 1996.01  5137.0 2000.16
  5167.6 2001.23  5188.0 2002.94  5218.6 2003.60  5239.0 2005.77  5259.4 2006.62
#Mann=3,-1,0
  4592.2    0.07       0  4994.7    0.05       0  5009.0    0.07       0
Bank Sta=4994.7,5009
Exp/Cntr=0.3,0.1
