HEC-RAS study Fessenden Branch.prj: Fessenden Branch Base Level Engineering

--- Fessenden Branch.g01 (geometry) --- (continued)

Type RM Length L Ch R = 1 ,22593   ,923,923,923
BEGIN DESCRIPTION:
Fessenden Branch 48.0
END DESCRIPTION:
XS GIS Cut Line= 3
      1860574.98     13979174.98        1860175.       13978775.
      1860074.99     13978674.99
#Sta/Elev= 30
  4438.6 2015.19  4466.9 2014.49  4551.7 2009.71  4650.7 2005.86  4735.6 2004.05
  4763.8  2004.2    4778 2003.54  4792.1 2003.78  4852.3 2003.42  4891.1 2003.09
  4905.3 2003.35  4919.4 2001.71  4933.6 1998.94  4947.7 1996.86  4961.8 1996.29
  4983.8 1996.05  4984.3 1995.55  4995.9 1995.55  4996.4 1996.05  5000.7 1996.46
  5018.4 1996.55  5032.5 1998.29  5044.9 1999.14  5046.7 1999.26  5060.8 2003.95
    5075 2007.54  5089.1 2009.13  5103.3 2010.23  5117.4 2010.06  5145.7 2010.69
#Mann= 5 ,-1 , 0
  4438.6      .1       0  4852.3     .07       0  4983.8     .05       0
  4996.4     .07       0  5044.9      .1       0
Bank Sta=4983.8,4996.4
XS Rating Curve= 0 ,0
Exp/Cntr=0.3,0.1

Type RM Length L Ch R = 1 ,21670   ,470,470,470
BEGIN DESCRIPTION:
Fessenden Branch 47.0
END DESCRIPTION:
XS GIS Cut Line= 3
      1861024.97     13978175.03        1860875.       13978325.
        1860175.       13978525.
#Sta/Elev= 30
  4789.1 2019.59  4803.2 2019.34  4817.3 2017.75  4863.2 2015.21  4916.3 2011.33
  4958.8 2006.16  4972.9 1995.55    4987 1989.45  4997.7 1987.39  5003.8 1987.39
  5004.3 1986.64  5004.8 1986.14  5018.9 1986.64  5032.4 1988.88  5042.8  1992.3
  5057.1 1993.51  5096.1 1993.61  5124.7  1995.7  5157.2 1995.79    5178 1997.06
  5212.9 1997.47  5241.4 1997.57  5270.3 1996.41  5316.4 1996.72  5348.3 1996.38
  5469.2 2000.34  5510.8  2000.4  5605.7 2002.57    5646 2004.92  5729.2 2006.07
#Mann= 7 ,-1 , 0
  4789.1      .1       0  4863.2     .07       0  5004.3     .05       0
  5018.9     .07       0  5212.9      .1       0  5241.4     .07       0
  5316.4      .1       0
Bank Sta=5004.3,5018.9
XS Rating Curve= 0 ,0
Exp/Cntr=0.3,0.1

Type RM Length L Ch R = 1 ,21200   ,384,384,384
BEGIN DESCRIPTION:
Fessenden Branch 46.0
END DESCRIPTION:
XS GIS Cut Line= 3
      1860775.02     13977924.99        1860575.       13977975.
      1859975.04     13978124.99
#Sta/Elev= 30
  4798.5 2011.21  4904.2 2007.38  4932.5 2004.22  4940.3 1998.37  4945.4 1988.78
  4953.1 1983.66  4966.5 1980.54    4967 1980.04  4981.1 1980.54  4994.5 1981.93
  5002.1  1984.4  5007.3  1984.4    5015 1986.79  5027.9 1989.06  5063.9  1990.3
  5080.6 1990.11  5138.7 1989.97  5151.6 1990.66  5187.6 1990.48  5200.5 1991.28
  5241.8 1988.58    5283 1991.39  5311.3 1992.16  5352.6 1991.98    5435 1996.85
  5447.9 1998.54  5476.3 2000.29  5489.1 2000.11  5558.7 2003.74  5623.1 2005.94
#Mann= 5 ,-1 , 0
  4798.5      .1       0  4966.5     .05       0  4981.1      .1       0
  4994.5     .07       0  5080.6      .1       0
Bank Sta=4966.5,4981.1
XS Rating Curve= 0 ,0
Exp/Cntr=0.3,0.1

Type RM Length L Ch R = 1 ,20816   ,186,186,186
BEGIN DESCRIPTION:
Fessenden Branch 45.0
END DESCRIPTION:
XS GIS Cut Line= 3
      1860533.25     13977673.91      1860280.39     13977784.47
      1859778.09      13977990.8
#Sta/Elev= 30
  4725.7 2002.92  4781.9 2001.74  4886.4 2000.16  4909.3 1996.44  4915.2 1994.87
  4920.7 1991.57  4944.1 1986.42    4962 1982.91  4977.9 1981.58  4978.4 1981.08
  4992.8 1981.58  4996.4 1982.78  5007.5 1983.04  5050.7 1982.15  5061.6 1983.18
  5067.9 1984.74  5073.3 1987.87  5083.2 1988.76  5145.2  1987.7  5158.9 1985.43
  5174.6 1984.67  5191.3 1987.12    5204 1990.97  5245.3 1996.16  5251.9 1998.12
  5281.3 2002.42  5329.2 2006.26  5406.6 2008.61  5465.3 2009.11  5544.7 2012.42
#Mann= 5 ,-1 , 0
  4725.7      .1       0  4781.9     .07       0  4977.9     .05       0
  4992.8     .07       0  5145.2      .1       0
Bank Sta=4977.9,4992.8
XS Rating Curve= 0 ,0
Exp/Cntr=0.3,0.1

Type RM Length L Ch R = 1 ,20630   ,321,321,321
BEGIN DESCRIPTION:
Mapping XS 2cc883fb
END DESCRIPTION:
XS GIS Cut Line= 2
      1860437.25     13977633.09      1859784.39     13977871.69
#Sta/Elev= 30
  4645.9 2000.88  4680.2 2001.12  4712.2 2000.16  4756.8 1996.67  4775.8 1993.09
    4782 1991.71  4818.6 1987.78  4837.7 1987.82    4843 1986.43  4893.2 1985.56
  4904.1 1983.81    4924 1984.03  4954.5 1982.67  4977.6 1977.97  4978.1 1977.47
  4992.5 1977.97  4999.6 1980.07  5040.8 1979.25  5046.2 1980.76  5063.5 1983.01
  5084.8 1991.28  5095.5 1993.35  5101.9  1996.2  5116.8 1999.55  5127.1 2001.66
    5170 2006.42  5188.2 2007.85    5224 2008.84  5311.8 2010.12    5341 2011.23
#Mann= 5 ,-1 , 0
  4645.9      .1       0  4775.8     .07       0  4977.6     .05       0
  4992.5     .07       0  5311.8      .1       0
Bank Sta=4977.6,4992.5
XS Rating Curve= 0 ,0
Exp/Cntr=0.3,0.1

Type RM Length L Ch R = 1 ,20309   ,251,251,251
BEGIN DESCRIPTION:
Fessenden Branch 44.0
END DESCRIPTION:
XS GIS Cut Line= 3
      1860424.96       13977575.        1859925.       13977525.
      1859724.95       13977525.
#Sta/Elev= 30
  4492.5 1999.12  4532.7 1998.66  4562.8 1996.45  4582.9 1993.91    4603 1992.51
  4633.2 1991.35  4723.6 1988.91  4733.7  1988.1  4753.8 1987.81  4763.8 1987.18
  4868.2 1986.45  4924.6 1984.94  4942.2 1983.54  4947.2 1984.66  4964.8 1979.79
  4974.9 1977.66    4995 1976.55  4997.5 1975.06    4998 1974.56    5012 1974.56
  5012.5 1975.06    5015 1975.41    5025 1988.49    5035 2000.34    5045 2004.71
    5055  2006.9    5075 2009.31    5095 2009.63    5115 2010.54    5195 2011.68
#Mann= 4 ,-1 , 0
  4492.5      .1       0  4868.2     .07       0  4997.5     .05       0
  5012.5      .1       0
Bank Sta=4997.5,5012.5
XS Rating Curve= 0 ,0
Exp/Cntr=0.3,0.1

Type RM Length L Ch R = 1 ,20058   ,199,199,199
BEGIN DESCRIPTION:
Mapping XS ff5965a5
END DESCRIPTION:
XS GIS Cut Line= 3
      1860576.24     13977488.56      1859869.74     13977290.74
      1859592.25     13977285.86
#Sta/Elev= 30
  4323.5 2002.91  4335.2 2001.95  4366.3 2001.04  4387.1 1999.49  4392.3 1998.44
  4480.6 1994.08  4646.7 1990.39  4698.6 1988.06  4719.4 1987.38  4740.2 1987.62
    4804 1985.17  4832.9 1985.04  4877.4 1986.67  4937.5 1984.71  4968.6 1981.17
    4979 1979.34    4985 1976.03  5010.2 1973.42  5011.6 1972.13  5012.1 1971.63
  5026.1 1971.63  5026.6 1972.13  5030.9 1984.71  5041.3 1994.41    5057 2007.06
  5086.9 2009.26  5103.2 2010.03  5151.9 2010.12  5221.9 2012.93  5334.7 2014.84
#Mann= 4 ,-1 , 0
  4323.5      .1       0  5011.6     .05       0  5026.6      .1       0
  5086.9     .07       0
#XS Ineff= 2 , 0
         4877.52 1986.34
Permanent Ineff=
       F       F
Bank Sta=5011.6,5026.6
XS Rating Curve= 0 ,0
Exp/Cntr=0.3,0.1

Type RM Length L Ch R = 1 ,19859   ,161,161,161
BEGIN DESCRIPTION:
Fessenden Branch 43.0
END DESCRIPTION:
XS GIS Cut Line= 3
      1860575.02     13977375.01        1859975.       13977125.
      1859775.03       13977125.
#Sta/Elev= 30
  4349.9 2002.17  4364.6 2001.92  4425.8 1995.48  4465.3 1992.81  4523.8 1991.93
  4571.5 1989.11  4609.9 1988.52  4642.4 1987.08  4685.8 1987.21  4718.3 1986.06
  4783.8 1985.45  4831.5    1984  4848.3 1982.53  4902.4 1983.68  4924.1  1983.3
  4961.5 1978.58  4967.4 1976.56  4985.3 1973.04  4999.9 1973.45  5002.4 1971.92
  5002.9 1971.42  5016.9 1971.42  5017.4 1971.92  5019.9 1972.26  5029.9 1985.24
  5049.9 2005.05  5059.9 2007.05  5069.9 2008.03  5092.3 2009.18  5199.9 2010.77
#Mann= 4 ,-1 , 0
  4349.9      .1       0  5002.4     .05       0  5017.4      .1       0
  5092.3     .07       0
#XS Ineff= 2 , 0
         4901.55 1983.81
Permanent Ineff=
       F       F
Bank Sta=5002.4,5017.4
XS Rating Curve= 0 ,0
Exp/Cntr=0.3,0.1

Type RM Length L Ch R = 1 ,19698   ,255,255,255
BEGIN DESCRIPTION:
Mapping XS 7e19f8cc
END DESCRIPTION:
XS GIS Cut Line= 3
      1860584.61     13977207.66      1859978.93     13976961.81
      1859722.01      13977005.6
#Sta/Elev= 30
  4429.9 2000.79  4432.4 2000.79    4448 1997.67  4483.4 1993.09  4515.8 1990.77
  4548.2 1990.23  4623.7  1985.8  4645.3 1986.11  4721.2 1984.13  4817.6 1983.72
  4900.6 1981.31  4924.7 1980.08  4936.7 1975.19  4940.7  1974.8  4947.5 1974.14
    4982 1975.24  5000.2 1972.99  5000.7 1972.49  5014.7 1972.49  5015.2 1972.99
  5031.8 1976.76  5037.2 1984.99  5044.6 1993.75  5055.4 2000.43  5061.3 2005.02
  5209.3 2008.62  5248.1 2008.84    5260  2009.6  5300.6 2009.66  5344.2 2010.98
#Mann= 4 ,-1 , 0
  4429.9      .1       0  4940.7     .07       0  5000.2     .05       0
  5015.2     .07       0
Bank Sta=5000.2,5015.2
XS Rating Curve= 0 ,0
Exp/Cntr=0.3,0.1

Type RM Length L Ch R = 1 ,19443   ,447,447,447
BEGIN DESCRIPTION:
Fessenden Branch 42.0
END DESCRIPTION:
XS GIS Cut Line= 3
        1860675.       13977025.        1860225.       13976825.
      1860025.04       13976825.
#Sta/Elev= 30
    4503 2001.93  4540.6 2000.84  4557.7 1998.11  4563.9 1996.32  4601.5 1992.37
  4623.4 1991.63  4633.6  1990.1  4656.2 1989.32  4685.6 1986.98  4714.3 1985.88
  4743.7 1983.28  4842.2 1981.48  4859.3 1980.25  4896.9 1979.15  4919.4 1976.86
  4940.7 1974.67  4963.3 1974.22  5007.9 1971.39  5008.4 1970.89  5022.5 1970.89
    5023 1971.39  5045.4 1975.16  5055.4 1984.87  5065.4 1990.42  5075.4 1993.42
  5085.4 1997.35  5095.4 2000.06  5105.4    2001  5135.4 2002.15  5195.4 2003.53
#Mann= 4 ,-1 , 0
    4503      .1       0  4919.4     .07       0  5007.9     .05       0
    5023     .07       0
Bank Sta=5007.9,5023
XS Rating Curve= 0 ,0
Exp/Cntr=0.3,0.1

Type RM Length L Ch R = 1 ,18996   ,449,449,449
BEGIN DESCRIPTION:
Fessenden Branch 41.0
END DESCRIPTION:
XS GIS Cut Line= 3
      1860825.03     13976675.02        1860525.       13976525.
      1860225.05       13976525.
#Sta/Elev= 30
  4664.8 2000.36  4695.6 1999.87  4745.9 1991.27  4807.4 1984.06  4835.3 1980.18
  4857.7 1978.36  4888.4 1977.12  4896.8 1977.18  4902.4 1976.51  4933.2 1975.07
  4941.6  1975.1  4955.5 1974.11  4977.9 1974.21  4986.3 1973.22  4989.8 1970.87
  4990.3 1970.37  5004.7 1970.37  5005.2 1970.87  5050.2 1972.38  5060.2 1971.04
  5090.2 1971.65  5100.2 1972.82  5110.2 1975.41  5120.2 1979.06  5130.2 1981.84
  5140.2 1983.09  5200.2 1987.36  5220.2 1989.88  5240.2 1990.17  5300.2 1993.76
#Mann= 3 ,-1 , 0
  4664.8      .1       0  4989.8     .05       0  5005.2      .1       0
Bank Sta=4989.8,5005.2
XS Rating Curve= 0 ,0
Exp/Cntr=0.3,0.1

Type RM Length L Ch R = 1 ,18547   ,426,426,426
BEGIN DESCRIPTION:
Fessenden Branch 40.0
END DESCRIPTION:
XS GIS Cut Line= 3
      1861024.97     13976224.99        1860775.       13976175.
      1860174.98     13975974.99
#Sta/Elev= 30
  4744.8  1999.9  4765.2 1999.48  4775.4 1998.68  4785.6 1996.86  4795.8 1993.18
    4806 1988.36  4816.2 1984.78  4826.4 1978.74  4836.6 1976.34    4857 1974.86
  4918.1 1973.87  4956.1 1971.49  4971.6 1969.88  4972.1 1969.38  4986.5 1969.38
    4987 1969.88  4989.5 1970.35  5010.3 1970.35  5031.3 1971.18  5052.4 1970.07
    5094 1971.42  5105.1 1971.43  5115.7 1973.77  5157.8    1977    5200 1979.17
  5252.7 1982.76  5294.9 1983.49    5337 1985.79  5537.3 1993.25  5632.2  1998.4
#Mann= 5 ,-1 , 0
  4744.8      .1       0  4956.1     .07       0  4971.6     .05       0
    4987     .07       0    5094      .1       0
Bank Sta=4971.6,4987
XS Rating Curve= 0 ,0
Exp/Cntr=0.3,0.1

Type RM Length L Ch R = 1 ,18121   ,448,448,448
BEGIN DESCRIPTION:
Fessenden Branch 39.0
END DESCRIPTION:
XS GIS Cut Line= 3
      1861175.01       13975875.        1860975.       13975825.
      1860375.04     13975725.01
#Sta/Elev= 30
  4793.5 2002.49  4845.1 2000.15    4876 1994.18  4899.2 1986.64  4906.9 1981.46
  4917.2 1976.69  4935.2 1969.71  4940.4 1968.74  4948.1 1967.66  4976.5 1967.41
  4989.4 1965.85  5002.1 1965.84  5002.6 1965.34  5017.5 1965.84  5027.5 1967.24
  5088.4 1968.25  5111.2 1971.51  5141.6 1973.18  5182.1 1972.47  5202.4 1970.65
  5215.1 1970.89  5222.7 1971.24    5243 1975.18  5303.8 1980.12  5336.8 1981.07
  5397.6  1984.7  5415.3 1984.57  5519.2 1988.99  5557.3 1991.41  5607.9 1993.01
#Mann= 3 ,-1 , 0
  4793.5      .1       0  5002.1     .05       0  5017.5      .1       0
Bank Sta=5002.1,5017.5
XS Rating Curve= 0 ,0
Exp/Cntr=0.3,0.1

Type RM Length L Ch R = 1 ,17673   ,371,371,371
BEGIN DESCRIPTION:
Fessenden Branch 38.0
END DESCRIPTION:
XS GIS Cut Line= 3
      1861225.01       13975425.        1861025.       13975425.
      1860574.98       13975475.
#Sta/Elev= 30
  4804.6 1990.99  4814.6 1990.29  4854.6 1989.87  4894.6 1986.56  4924.6 1981.56
  4944.6 1975.39  4954.6 1970.18  4964.6 1962.04  4976.9 1957.88  4977.4 1957.38
  4991.8 1957.38  4992.3 1957.88  4994.6 1959.92  5007.1 1959.81  5054.9 1967.73
  5085.1 1969.83  5105.2 1970.12  5145.5 1969.09  5185.7 1966.88  5195.8 1966.78
  5215.9 1968.96    5236 1969.05  5256.1 1970.45  5306.5 1971.73  5316.5  1972.4
  5326.6 1974.05  5346.7  1976.2  5407.1 1981.44  5437.3 1983.28  5457.4 1983.27
#Mann= 3 ,-1 , 0
  4804.6      .1       0  4976.9     .05       0  4992.3      .1       0
Bank Sta=4976.9,4992.3
XS Rating Curve= 0 ,0
Exp/Cntr=0.3,0.1

Type RM Length L Ch R = 1 ,17302   ,202,202,202
BEGIN DESCRIPTION:
Fessenden Branch 37.0
END DESCRIPTION:
XS GIS Cut Line= 3
        1861125.       13975075.      1860746.61     13975096.22
      1860474.98     13974874.99
#Sta/Elev= 30
  4799.6 1983.53  4849.7 1982.87  4879.7 1980.16  4886.8 1978.06  4891.8 1978.05
  4899.8 1975.22  4909.8 1973.05  4919.8 1971.89  4929.8 1969.59  4949.8 1961.74
  4959.8 1958.64  4982.1 1955.98  4982.6 1955.48  4997.6 1955.98  4999.9 1957.03
  5019.9 1959.33    5080 1961.73  5110.1 1965.37  5150.1 1966.82  5187.8 1970.25
  5194.2 1969.53  5237.3 1970.66  5315.6  1975.6  5379.5 1983.62  5408.2 1988.35
  5443.4 1991.78  5472.2 1997.95    5493 1999.83  5500.9 2001.31  5528.9 2002.82
#Mann= 3 ,-1 , 0
  4799.6      .1       0  4982.1     .05       0  4997.6      .1       0
Bank Sta=4982.1,4997.6
XS Rating Curve= 0 ,0
Exp/Cntr=0.3,0.1

Type RM Length L Ch R = 1 ,17100   ,43,43,43
BEGIN DESCRIPTION:
Fessenden Branch 36.1
END DESCRIPTION:
XS GIS Cut Line= 4
      1861175.26     13974961.48      1860896.18     13974940.99
      1860677.66     13974945.08      1860532.23     13974897.51
#Sta/Elev= 30
    4648 1980.12  4718.5 1979.61  4728.5 1977.43  4738.5  1973.9  4758.6 1971.98
  4798.7 1971.35  4818.7 1967.66  4858.8  1967.7  4868.9 1964.94  4888.9 1961.58
  4898.9 1960.61  4941.3 1959.65  4941.8 1959.15  4956.8 1959.65    4959  1960.8
    5009 1959.74    5099  1961.4    5109 1964.97  5132.3    1970  5145.2 1972.03
  5163.8 1972.62  5190.5 1977.24  5195.7 1977.11  5212.3 1982.13  5243.9 1987.68
  5259.4 1989.42  5264.9 1990.94    5286 1993.21  5291.3 1995.18  5299.4 1996.01
#Mann= 4 ,-1 , 0
    4648     .07       0  4941.3     .05       0  4956.8     .07       0
  5132.3      .1       0
Bank Sta=4941.3,4956.8
XS Rating Curve= 0 ,0
Exp/Cntr=0.3,0.1

Type RM Length L Ch R = 1 ,17057   ,65,65,65
BEGIN DESCRIPTION:
Fessenden Branch 36.2
END DESCRIPTION:
XS GIS Cut Line= 5
      1861283.18     13974902.46      1860929.44     13974893.78
      1860817.67     13974904.63      1860771.01     13974905.72
      1860515.99     13974862.31
#Sta/Elev= 30
  4520.5 1980.28  4558.7 1980.33  4628.7 1978.32  4658.7 1974.78  4688.7 1973.01
  4708.7 1971.03  4728.7 1970.93    4741 1967.65  4741.5 1967.15    4756 1967.15
  4756.5 1967.65  4768.8 1967.99  4798.8  1967.7  4838.8 1969.47  4848.8 1974.58
  4858.8 1975.51  4888.9 1974.92  4936.4    1975  4941.4 1974.31  4979.3 1974.27
  5071.1 1975.57  5126.3 1977.48  5131.4 1975.47    5151 1977.43  5161.1  1978.9
  5181.4 1982.18  5186.5 1984.42    5227 1990.49  5272.7 1998.68    5292 2000.46
#Mann= 4 ,-1 , 0
  4520.5     .07       0    4741     .05       0  4756.5     .07       0
    5227      .1       0
#XS Ineff= 2 , 0
                         4860.54         1975.62
Permanent Ineff=
       F       F
Bank Sta=4741,4756.5
XS Rating Curve= 0 ,0
Exp/Cntr=0.3,0.1

Type RM Length L Ch R = 1 ,16992   ,638,638,638
BEGIN DESCRIPTION:
Fessenden Branch 35.1
END DESCRIPTION:
XS GIS Cut Line= 4
      1861292.43     13974851.86      1861119.09      13974838.9
      1860634.76     13974854.68       1860519.4     13974804.05
#Sta/Elev= 30
  4481.5 1976.63  4505.2 1976.05  4510.2 1974.82  4539.1 1976.67  4589.2  1973.3
  4699.4 1970.56  4709.4 1968.36  4729.5 1967.66  4769.5 1969.46  4799.5 1976.85
  4809.5 1974.46  4829.5 1962.82  4919.6 1962.71  4929.6  1961.7  4931.8 1960.08
  4932.3 1959.58  4947.4 1960.08  4959.6 1962.19  4979.6 1962.88  4989.6 1962.12
  4995.4 1960.25  5009.6 1962.77  5019.6 1961.51  5119.7  1977.6  5137.3  1982.2
  5142.5  1982.2  5148.3 1984.25  5194.3 1992.03  5237.9 2001.07  5265.9 2004.02
#Mann= 3 ,-1 , 0
  4481.5     .07       0  4931.8     .05       0  4947.4     .07       0
#XS Ineff= 2 , 0
         4796.64  1976.1
Permanent Ineff=
       F       F
Bank Sta=4931.8,4947.4
XS Rating Curve= 0 ,0
Exp/Cntr=0.3,0.1

Type RM Length L Ch R = 1 ,16354   ,457,457,457
BEGIN DESCRIPTION:
Fessenden Branch 35.0
END DESCRIPTION:
XS GIS Cut Line= 3
      1861301.17     13974828.03        1860975.       13974325.
      1860774.98     13974274.99
#Sta/Elev= 30
    4391    1974  4418.4 1971.94  4490.5 1969.73  4549.5 1964.86  4608.5  1964.2
  4629.6 1962.01  4702.1 1960.98  4729.1 1963.07  4765.4 1962.92  4795.7  1960.9
  4801.7 1962.51  4890.2 1958.18  4925.6 1955.19  4940.7  1955.3    4977 1951.24
  4982.9 1952.57    4993 1950.83  4993.5 1950.33  5008.6 1950.83  5031.8  1959.6
  5049.8 1969.29  5054.9 1978.11  5061.2  1984.9  5062.7 1986.52  5083.3 1992.08
    5091 1996.19  5096.2 2000.54  5103.9 2002.37  5155.4 2008.79  5196.7 2010.93
#Mann= 5 ,-1 , 0
    4391     .07       0  4890.2      .1       0    4993     .05       0
  5008.6      .1       0  5061.2     .07       0
#XS Ineff= 2 , 0
          4800.4 1962.85
Permanent Ineff=
       F       F
Bank Sta=4993,5008.6
XS Rating Curve= 0 ,0
Exp/Cntr=0.3,0.1

Type RM Length L Ch R = 1 ,15897   ,480,480,480
BEGIN DESCRIPTION:
Fessenden Branch 34.0
END DESCRIPTION:
XS GIS Cut Line= 3
        1861425.     13974874.99        1861375.       13974275.
        1861225.       13974125.
#Sta/Elev= 30
    4398 1979.44  4428.1  1977.3    4451 1974.52  4511.6 1970.97  4538.5 1969.75
  4576.1 1964.71  4581.1 1964.97  4598.7 1962.94  4648.9 1959.78  4829.5 1956.22
  4849.6 1954.78  4859.6 1952.59  4879.7 1954.95  4919.8  1954.5  4937.4 1953.16
  4959.9 1949.73    4980 1948.49  4989.8 1946.07  4990.3 1945.57  5005.4 1946.07
  5032.3 1947.08  5056.6 1948.86  5070.8  1953.1  5084.9 1960.14  5113.2 1984.28
  5130.3 1988.17  5141.5 1989.93  5155.6 1993.67  5169.8 1995.76  5212.2  1997.5
#Mann= 7 ,-1 , 0
    4398     .07       0    4451      .1       0  4511.6     .07       0
  4989.8     .05       0  5005.4     .07       0  5032.3      .1       0
  5130.3     .07       0
#XS Ineff= 2 , 0
         4882.12 1955.09
Permanent Ineff=
       F       F
Bank Sta=4989.8,5005.4
XS Rating Curve= 0 ,0
Exp/Cntr=0.3,0.1

Type RM Length L Ch R = 1 ,15417   ,143,143,143
BEGIN DESCRIPTION:
Fessenden Branch 33.0
END DESCRIPTION:
XS GIS Cut Line= 3
      1861500.26     13974891.97        1861825.       13974375.
      1861774.99     13974174.96
#Sta/Elev= 30
  4383.7 1978.52  4421.1 1978.57  4442.3 1975.92  4478.9 1974.21  4509.5  1970.7
  4594.3 1967.17  4609.6 1965.88  4624.9 1963.16  4630.8 1963.48  4646.1 1961.21
  4668.4 1959.73  4703.8 1956.73  4719.1 1954.15  4840.7 1952.46  4907.6 1949.19
  4928.8 1949.12  4944.1 1946.65  4958.8 1945.66  4980.6 1945.95  4991.2 1944.23
  5004.4 1943.96  5004.9 1943.46    5020 1943.96  5045.7 1950.12  5053.5 1954.75
  5058.6 1954.28  5066.4 1957.59  5095.1  1966.2  5135.9 1967.55  5200.4 1973.76
#Mann= 5 ,-1 , 0
  4383.7      .1       0  4668.4     .07       0  5004.4     .05       0
    5020     .07       0  5095.1      .1       0
Bank Sta=5004.4,5020
XS Rating Curve= 0 ,0
Exp/Cntr=0.3,0.1

Type RM Length L Ch R = 1 ,15274   ,310,310,310
BEGIN DESCRIPTION:
Mapping XS bf798c70
END DESCRIPTION:
XS GIS Cut Line= 3
        1861965.     13974941.53      1861953.22      13974443.3
      1861839.69     13974081.05
#Sta/Elev= 30
  4482.1 1980.35  4518.6 1978.13  4618.7 1966.01  4628.7  1964.2  4658.7 1954.47
  4668.7 1952.57  4713.5 1952.24  4888.7 1951.26  4948.8 1945.82  4987.6 1945.09
  4992.8 1945.81  5017.3 1944.89  5017.8 1944.39  5033.3 1944.89  5041.6 1945.99
    5073 1946.26  5083.5 1947.18  5090.1 1948.71  5095.4 1948.62  5122.6 1955.93
  5127.8 1956.23  5140.4 1959.06    5155 1961.86  5160.3 1961.81  5177.8 1965.72
  5192.7  1967.1  5219.7 1967.53  5240.7 1968.78  5327.7 1976.17  5360.1 1976.76
#Mann= 5 ,-1 , 0
  4482.1      .1       0  4713.5     .07       0  5017.3     .05       0
  5033.3     .07       0  5140.4      .1       0
Bank Sta=5017.3,5033.3
XS Rating Curve= 0 ,0
Exp/Cntr=0.3,0.1

Type RM Length L Ch R = 1 ,14964   ,464,464,464
BEGIN DESCRIPTION:
Fessenden Branch 32.0
END DESCRIPTION:
XS GIS Cut Line= 3
        1862125.       13974925.        1862225.       13974525.
      1861925.01     13973975.01
#Sta/Elev= 30
  4588.1 1981.86  4639.6 1977.67    4686 1969.36  4711.8 1965.71  4722.1 1963.02
  4729.8 1959.32    4735 1958.15  4742.7 1954.81  4763.3  1949.9  4771.1 1949.25
  4866.4 1949.02  4977.2 1950.12  4990.1 1949.28  4997.8 1946.91  5003.3 1946.91
  5008.5 1944.66  5014.2 1944.81  5015.2 1942.88  5015.7 1942.38  5031.2 1942.88
    5036 1944.38    5046 1944.92  5161.3 1944.99  5205.4 1951.43  5261.8 1954.73
  5324.6  1957.2  5411.9 1966.35  5471.7 1967.83  5575.2 1974.62  5626.9 1976.64
#Mann= 5 ,-1 , 0
  4588.1      .1       0    4686     .07       0  5015.2     .05       0
  5031.2     .07       0  5261.8      .1       0
Bank Sta=5015.2,5031.2
XS Rating Curve= 0 ,0
Exp/Cntr=0.3,0.1

Type RM Length L Ch R = 1 ,14500   ,370,370,370
BEGIN DESCRIPTION:
Fessenden Branch 31.0
END DESCRIPTION:
XS GIS Cut Line= 3
        1862675.     13974675.02        1862675.       13974475.
      1862325.03     13973975.04
#Sta/Elev= 30
  4795.3 1991.77  4855.3 1990.76  4895.3  1986.4  4907.9 1983.29  4915.3 1980.45
  4925.3 1974.49  4935.3 1969.88  4945.3    1962  4955.3 1956.38  4984.7 1937.83
  4985.2 1937.33  5000.9 1937.83  5002.7 1938.65  5017.6 1939.35  5031.9  1943.4
  5074.2 1944.51  5089.1 1945.95  5117.4 1947.18  5190.2 1946.57  5202.8  1947.2
  5246.9 1945.65  5261.7 1947.58  5419.5 1952.57  5470.1 1955.35  5511.9 1959.36
  5547.7 1964.25  5583.4 1966.31  5592.1 1966.19  5598.2 1967.26  5605.6 1966.99
#Mann= 4 ,-1 , 0
  4795.3      .1       0  4907.9     .07       0  4984.7     .05       0
  5000.9     .07       0
Bank Sta=4984.7,5000.9
XS Rating Curve= 0 ,0
Exp/Cntr=0.3,0.1

Type RM Length L Ch R = 1 ,14130   ,494,494,494
BEGIN DESCRIPTION:
Fessenden Branch 30.0
END DESCRIPTION:
XS GIS Cut Line= 3
      1862979.88     13974476.38      1862960.25     13974243.87
      1862374.99       13973975.
#Sta/Elev= 30
  4725.5 1984.96  4777.1 1984.27  4816.2 1981.25  4837.3  1977.4  4842.6  1975.3
  4847.6 1975.92  4887.5 1969.45  4917.6 1958.85  4937.6 1954.13  4958.8 1950.63
  4975.6 1936.68    4984  1934.7  4984.5  1934.2  5000.2  1934.7  5015.1 1936.65
  5038.1 1942.64    5107 1945.22  5135.5  1945.4  5173.7 1942.99  5195.7  1942.8
  5217.7 1943.36  5239.7 1945.25  5316.8 1946.65  5370.8 1949.47  5399.3 1949.67
  5491.2 1954.53  5525.9 1959.57  5548.2 1961.31  5571.2 1964.44  5602.9 1965.39
#Mann= 4 ,-1 , 0
  4725.5      .1       0  4816.2     .07       0    4984     .05       0
  5000.2     .07       0
Bank Sta=4984,5000.2
XS Rating Curve= 0 ,0
Exp/Cntr=0.3,0.1

Type RM Length L Ch R = 1 ,13636   ,484,484,484
BEGIN DESCRIPTION:
Fessenden Branch 29.0
END DESCRIPTION:
XS GIS Cut Line= 4
      1863725.87     13973926.57      1863346.61      13973867.9
        1863175.       13973825.      1862374.96       13973825.
#Sta/Elev= 30
  4439.4 2006.46    4501  2006.7  4547.2 2004.04  4622.4 2003.58  4774.2 1997.03
  4809.5 1993.23  4821.5 1988.16  4826.6 1988.16  4845.4 1977.53  4853.2 1971.37
  4858.3 1969.48  4866.1 1962.36  4887.5 1950.72  4894.4  1945.5  4899.6 1944.03
  4907.3 1939.25  4917.6 1936.11  4969.1  1935.1  4976.9 1934.32  4981.3 1930.57
  4981.8 1930.07  4998.2 1930.57  5040.1 1938.79  5108.4 1941.59  5163.8 1942.79
  5350.1  1941.8  5480.1 1944.41  5620.1 1950.76  5750.1 1965.45  5800.1 1966.89
#Mann= 6 ,-1 , 0
  4439.4      .1       0  4887.5     .07       0  4981.3     .05       0
  4998.2     .07       0  5108.4      .1       0  5163.8     .07       0
Bank Sta=4981.3,4998.2
XS Rating Curve= 0 ,0
Exp/Cntr=0.3,0.1

Type RM Length L Ch R = 1 ,13152   ,447,447,447
BEGIN DESCRIPTION:
Fessenden Branch 28.0
END DESCRIPTION:
XS GIS Cut Line= 3
        1863375.       13973375.        1863175.       13973375.
      1862575.01     13973774.99
#Sta/Elev= 30
  4805.1 2002.89  4845.1 2001.49  4855.1 2000.23  4875.1 1995.15  4885.1 1991.13
  4915.1 1976.29  4925.1 1969.16  4935.1 1958.56  4945.1 1943.82    4963 1933.82
  4975.1 1928.02  4986.6  1924.7  4987.1  1924.2  5003.6  1924.7  5005.1 1927.09
  5008.1 1927.09  5027.6 1932.38  5054.7 1934.14  5077.2 1934.34  5090.7 1936.57
  5113.3 1938.22  5154.5 1938.88  5288.5 1938.67  5379.2 1938.25  5517.4 1942.06
  5610.5 1943.35  5631.6 1945.07  5658.2 1945.44  5710.6  1948.5  5726.2 1949.35
#Mann= 8 ,-1 , 0
  4805.1      .1       0    4963     .07       0  4986.6     .05       0
  5003.6     .07       0  5154.5      .1       0  5288.5     .07       0
  5658.2      .1       0  5710.6     .07       0
Bank Sta=4986.6,5003.6
XS Rating Curve= 0 ,0
Exp/Cntr=0.3,0.1

Type RM Length L Ch R = 1 ,12705   ,507,507,507
BEGIN DESCRIPTION:
Fessenden Branch 27.0
END DESCRIPTION:
XS GIS Cut Line= 3
      1863075.03     13973024.99        1862875.       13973075.
      1862274.99     13973525.01
#Sta/Elev= 30
  4793.8 1977.88  4818.2 1974.11  4824.8 1972.28  4835.1 1967.87  4853.1 1956.07
  4858.3 1950.81    4866 1945.63  4894.3 1931.83  4917.5 1927.82  4958.4  1926.6
  4981.2 1925.97  4981.7 1925.47  4998.2 1925.97  5007.3 1926.65  5013.5 1928.75
  5042.7 1932.84    5050 1932.38  5075.1 1933.31  5121.9  1933.6  5171.9 1935.41
  5348.3 1936.69  5407.3  1938.8  5436.4 1938.95  5486.4 1942.25  5607.3 1952.35
  5642.7 1953.92  5686.4 1958.68  5721.9 1964.45  5736.4 1965.71    5750 1965.44
#Mann= 7 ,-1 , 0
  4793.8      .1       0  4818.2     .07       0  4958.4      .1       0
  4981.2     .05       0  4998.2      .1       0  5075.1     .07       0
  5348.3      .1       0
Bank Sta=4981.2,4998.2
XS Rating Curve= 0 ,0
Exp/Cntr=0.3,0.1

Type RM Length L Ch R = 1 ,12198   ,362,362,362
BEGIN DESCRIPTION:
Fessenden Branch 26.0
END DESCRIPTION:
XS GIS Cut Line= 3
        1862875.       13972475.      1862502.83     13972802.21
      1861974.98     13973025.01
#Sta/Elev= 30
  4503.5 1972.91  4545.7 1968.32  4581.8 1961.42  4794.3  1938.2  4815.2 1933.98
  4829.4 1932.69  4843.6 1934.22  4850.3 1932.78  4857.9 1933.68  4864.5 1931.99
  4872.1 1932.78  4878.8 1930.67  4907.2 1928.11    4929 1923.74    4948 1923.27
  4948.5 1922.77  4965.2 1923.27  4997.4 1924.16  5029.3 1926.88  5309.7 1931.75
  5375.1 1931.69  5398.3 1933.56    5420 1939.37  5436.3 1946.58  5463.4 1954.18
    5496  1959.3  5517.7 1965.55  5533.7 1967.15  5539.4 1969.15    5572 1970.91
#Mann= 4 ,-1 , 0
  4503.5     .07       0    4948     .05       0  4965.2     .07       0
  5309.7      .1       0
Bank Sta=4948,4965.2
XS Rating Curve= 0 ,0
Exp/Cntr=0.3,0.1

Type RM Length L Ch R = 1 ,11836   ,485,485,485
BEGIN DESCRIPTION:
Fessenden Branch 25.0
END DESCRIPTION:
XS GIS Cut Line= 3
      1862825.02     13972374.99        1862225.       13972575.
      1861874.97       13972575.
#Sta/Elev= 30
  4374.9 1971.77  4427.6 1962.62    4533 1949.61  4606.8 1941.52  4627.9 1938.43
  4691.1 1934.63  4754.4 1932.24  4828.2 1931.59    4923 1929.48  4933.6 1925.69
  4954.7  1921.3  4986.3 1919.18  4996.1 1917.45  4996.6 1916.95  5013.4 1917.45
  5037.4 1921.91  5057.4 1922.03  5097.4 1925.01  5147.4 1926.43  5177.4 1924.88
  5197.4 1922.26  5207.4 1925.16  5237.7 1925.68  5257.4 1927.61  5267.4 1930.68
  5287.4 1941.06  5317.4 1962.25  5327.4 1970.11  5337.4 1975.12  5357.4 1977.46
#Mann= 4 ,-1 , 0
  4374.9     .07       0  4996.1     .05       0  5013.4     .07       0
  5237.7      .1       0
#XS Ineff= 2 , 0
                         5143.46         1926.21
Permanent Ineff=
       F       F
Bank Sta=4996.1,5013.4
XS Rating Curve= 0 ,0
Exp/Cntr=0.3,0.1

Type RM Length L Ch R = 1 ,11351   ,445,445,445
BEGIN DESCRIPTION:
Fessenden Branch 24.0
END DESCRIPTION:
XS GIS Cut Line= 3
      1862764.27     13972208.15        1862025.       13972175.
      1861825.01       13972175.
#Sta/Elev= 30
  4259.6 1962.61  4268.9 1961.13  4288.9 1960.16  4437.8 1941.74  4479.1 1938.67
  4539.2 1932.47  4609.2 1929.22  4639.3 1929.98  4759.4 1928.07  4819.4 1926.36
  4849.5 1924.54  4886.2 1925.07  4909.5 1924.11  4949.6 1919.89  4959.6 1916.67
  4999.6 1909.81    5001 1908.33  5001.5 1907.83  5018.3 1908.33  5019.6 1932.53
  5029.6 1946.62  5039.6 1953.62  5059.6 1962.83  5069.6 1968.93  5079.6 1972.36
  5099.6  1975.3  5119.6 1976.89  5159.6 1984.23  5169.6  1985.4  5199.6 1985.43
#Mann= 3 ,-1 , 0
  4259.6     .07       0    5001     .05       0  5018.3     .07       0
Bank Sta=5001,5018.3
XS Rating Curve= 0 ,0
Exp/Cntr=0.3,0.1

Type RM Length L Ch R = 1 ,10906   ,476,476,476
BEGIN DESCRIPTION:
Fessenden Branch 23.0
END DESCRIPTION:
XS GIS Cut Line= 3
      1862624.96     13971675.01        1862175.       13971775.
      1861974.99       13971825.
#Sta/Elev= 30
  4533.1 1954.94  4557.4 1953.58  4600.9 1946.33    4606 1946.69  4644.5 1938.55
  4649.6 1938.75    4656 1935.94  4693.1 1929.67  4698.2 1930.21  4736.7 1924.26
  4778.9 1923.94  4785.3 1922.58    4834 1920.92  4860.9 1917.27  4882.6 1918.48
  4932.6 1917.86  4953.1 1917.12  4969.7 1914.18  5008.5 1913.21    5009 1912.71
  5025.9 1913.21  5045.6 1919.07  5053.3 1925.16  5058.5 1923.21  5066.2  1931.5
  5094.5 1946.68  5099.7 1946.27  5135.8 1956.16  5182.2  1960.9  5200.2  1965.5
#Mann= 3 ,-1 , 0
  4533.1     .07       0  5008.5     .05       0  5025.9     .07       0
Bank Sta=5008.5,5025.9
XS Rating Curve= 0 ,0
Exp/Cntr=0.3,0.1

Type RM Length L Ch R = 1 ,10430   ,385,385,385
BEGIN DESCRIPTION:
Fessenden Branch 22.0
END DESCRIPTION:
XS GIS Cut Line= 3
      1862624.96     13971474.99        1862375.       13971375.
      1861924.96     13971575.02
#Sta/Elev= 30
  4731.2  1954.5  4763.5 1951.16  4799.8 1942.94  4824.1 1932.48  4848.3 1925.83
  4871.2 1921.88    4956 1918.93  4968.1 1917.54  4978.9 1914.52  4985.6  1911.2
  5006.1 1910.15  5006.6 1909.65  5023.5 1910.15  5032.6 1911.93  5045.2 1912.58
  5055.1  1912.1  5113.3 1915.08  5120.3 1914.28  5136.5 1913.82  5175.5 1915.68
    5183 1917.38  5188.5 1916.43  5206.3  1920.6  5229.5 1922.03    5235 1921.34
  5295.9 1926.58  5350.6 1933.41  5394.4 1942.27  5438.1 1949.61  5492.9 1955.03
#Mann= 5 ,-1 , 0
  4731.2     .07       0  5006.1     .05       0  5023.5     .07       0
  5045.2    .035       0  5120.3     .07       0
Bank Sta=5006.1,5023.5
XS Rating Curve= 0 ,0
Exp/Cntr=0.3,0.1

Type RM Length L Ch R = 1 ,10045   ,585,585,585
BEGIN DESCRIPTION:
Fessenden Branch 21.0
END DESCRIPTION:
XS GIS Cut Line= 3
      1862637.81     13970805.19      1862335.12     13970997.86
      1861825.03     13971424.98
#Sta/Elev= 30
  4627.8 1978.71  4658.1 1977.79  4666.7 1975.64  4694.5 1965.48  4724.9 1958.55
    4752 1948.98  4767.1 1941.06  4801.3 1918.59  4803.7  1916.8  4809.6 1916.42
  4818.9 1912.71  4832.6 1910.33  4855.3 1910.95  4891.7 1908.58    5004  1907.2
  5004.5  1906.7  5021.7  1907.2  5034.5 1913.08  5041.1  1912.1  5045.6 1915.16
  5048.8 1917.34  5055.4 1916.84  5077.5 1920.13  5159.7 1920.77  5219.3 1920.03
  5303.6 1921.27  5417.2 1924.15  5488.6 1932.78  5573.7  1946.9  5651.9 1951.82
#Mann= 8 ,-1 , 0
  4627.8      .1       0  4767.1     .07       0  4801.3     .07       0
    5004     .05       0  5021.7     .07       0  5045.6     .07       0
  5159.7      .1       0  5303.6     .07       0
Bank Sta=5004,5021.7
XS Rating Curve= 0 ,0
Exp/Cntr=0.3,0.1

Type RM Length L Ch R = 1 ,9460    ,448,448,448
BEGIN DESCRIPTION:
Fessenden Branch 20.0
END DESCRIPTION:
XS GIS Cut Line= 3
      1862175.01     13970325.03        1862225.       13970525.
      1862040.06     13971130.25
#Sta/Elev= 30
  4794.4 1998.86  4845.9 1996.73  4876.8 1993.95  4894.9 1994.09    4900 1992.52
  4918.1 1990.93  4928.4 1988.58  4936.1 1984.46  4941.3 1984.15    4949 1980.47
  4969.6 1955.77  4977.3 1909.13  4982.5 1909.18  4997.9  1902.7  5003.1  1902.7
    5011 1895.38  5013.3  1895.3  5013.8  1894.8    5031  1895.3  5049.7  1901.7
  5054.9 1901.39  5063.3 1903.95  5105.1 1910.68  5153.3 1913.52  5218.9 1914.92
  5327.8  1914.5  5408.3 1917.31  5495.6 1916.94  5567.8 1917.83  5633.4 1920.47
#Mann= 4 ,-1 , 0
  4794.4     .07       0  5013.3     .05       0    5031     .07       0
  5495.6      .1       0
#XS Ineff= 2 , 0
                         5165.83         1914.97
Permanent Ineff=
       F       F
Bank Sta=5013.3,5031
XS Rating Curve= 0 ,0
Exp/Cntr=0.3,0.1

Type RM Length L Ch R = 1 ,9012    ,446,446,446
BEGIN DESCRIPTION:
Fessenden Branch 19.0
END DESCRIPTION:
XS GIS Cut Line= 3
      1861875.01     13970474.97        1861825.       13970675.
        1861725.       13971225.
#Sta/Elev= 30
  4793.5 1988.68  4796.1 1988.68  4845.1 1967.39  4852.8  1962.5  4872.9 1953.89
  4886.3 1948.13    4894  1942.8  4906.9  1938.3  4917.2 1932.21  4935.3 1907.54
  4940.4 1911.06  4948.1 1902.39  4958.5 1897.82  5000.9 1895.05  5001.4 1894.55
  5018.7 1895.05  5025.1  1898.3  5050.5 1903.05  5118.4 1905.09  5191.5 1909.12
  5282.8 1909.24  5355.4 1909.86  5385.9 1912.35  5420.2 1921.73  5426.6 1925.58
  5446.9 1933.09  5467.2 1936.78  5479.6 1936.35  5526.9 1944.99  5558.7  1946.4
#Mann= 7 ,-1 , 0
  4793.5      .1       0  4872.9     .07       0  5000.9     .05       0
  5018.7     .07       0  5118.4      .1       0  5282.8    .035       0
  5479.6     .07       0
#XS Ineff= 2 , 0
         4939.66 1910.66 5186.41         1909.22
Permanent Ineff=
       F       F
Bank Sta=5000.9,5018.7
XS Rating Curve= 0 ,0
Exp/Cntr=0.3,0.1

Type RM Length L Ch R = 1 ,8566    ,482,482,482
BEGIN DESCRIPTION:
Fessenden Branch 18.0
END DESCRIPTION:
XS GIS Cut Line= 3
      1861324.99     13970424.98        1861425.       13970825.
      1861525.01     13971125.04
#Sta/Elev= 30
  4583.1 1997.02  4606.3 1992.57    4616 1989.29  4642.4 1979.63  4647.5 1979.41
  4683.6 1960.84  4688.8 1960.73  4706.8 1952.09  4717.1 1948.77  4766.1 1924.86
  4771.2 1924.15  4789.3 1914.92  4808.8 1909.81  4840.8 1906.05  4936.2  1901.8
  4977.4 1895.01    4984 1891.55  4984.5 1891.05  5001.8 1891.55  5027.1 1892.76
  5048.3 1896.56  5069.2 1897.31  5090.3 1900.06  5164.1 1902.65  5195.7 1906.77
  5215.1 1910.99  5237.9 1917.19    5280 1931.86  5304.9  1933.9  5311.7 1934.38
#Mann= 8 ,-1 , 0
  4583.1     .07       0    4616      .1       0  4808.8     .07       0
    4984     .05       0  5001.8     .07       0  5048.3    .035       0
  5215.1     .07       0  5304.9    .035       0
Bank Sta=4984,5001.8
XS Rating Curve= 0 ,0
Exp/Cntr=0.3,0.1

Type RM Length L Ch R = 1 ,8084    ,456,456,456
BEGIN DESCRIPTION:
Fessenden Branch 17.0
END DESCRIPTION:
XS GIS Cut Line= 3
        1860875.     13970575.01        1860975.       13970925.
      1861124.98     13971074.98
#Sta/Elev= 30
  4635.9 1979.72  4646.3 1979.41  4664.1 1973.98  4686.6 1964.85  4691.8 1964.25
  4698.3 1960.19  4719.1 1953.17  4725.6 1948.38  4730.8 1947.33  4750.3 1936.86
  4759.4  1931.5  4764.6 1926.85  4803.6 1908.88  4823.1 1903.68  4837.4 1901.27
  4848.3 1900.58  4910.2 1898.01  4958.3 1892.23  4977.8 1890.43    4983 1890.83
  4989.5 1889.29  5005.1 1888.81  5005.6 1888.31  5022.9 1888.81  5042.3 1888.81
  5056.5 1890.12  5070.6 1893.01  5098.9 1905.06    5113  1908.8    5212 1913.03
#Mann= 5 ,-1 , 0
  4635.9     .07       0  4664.1      .1       0  4848.3     .07       0
  5005.1     .05       0  5022.9     .07       0
Bank Sta=5005.1,5022.9
XS Rating Curve= 0 ,0
Exp/Cntr=0.3,0.1

Type RM Length L Ch R = 1 ,7628    ,459,459,459
BEGIN DESCRIPTION:
Fessenden Branch 16.0
END DESCRIPTION:
XS GIS Cut Line= 3
        1860575.     13970775.05        1860575.       13970975.
      1861025.03     13971575.04
#Sta/Elev= 30
  4800.4 1957.73  4880.4 1954.73  4900.4  1950.4  4910.4 1945.37  4930.4 1930.31
  4940.4 1919.63  4950.4 1912.08  4960.4 1897.05  4981.5 1887.83    4982 1887.33
  4999.3 1887.83  5078.5 1890.49  5086.8 1893.33  5100.4 1894.91  5107.6 1896.82
  5143.1 1896.31  5272.2 1899.03  5293.1 1901.04  5313.9 1904.67  5363.9 1908.14
  5422.2 1910.82  5478.5 1918.05  5486.8 1918.14  5550.4 1925.58  5622.2 1931.77
  5657.6 1937.26  5663.9 1937.44  5707.6 1944.85  5736.8  1947.8  5750.4 1948.12
#Mann= 3 ,-1 , 0
  4800.4     .07       0  4981.5     .05       0  4999.3     .07       0
Bank Sta=4981.5,4999.3
XS Rating Curve= 0 ,0
Exp/Cntr=0.3,0.1

Type RM Length L Ch R = 1 ,7169    ,419,419,419
BEGIN DESCRIPTION:
Fessenden Branch 15.0
END DESCRIPTION:
XS GIS Cut Line= 3
        1860225.       13971075.        1860275.       13971275.
      1860525.01     13971775.02
#Sta/Elev= 30
  4793.4 1937.06  4816.6 1933.61  4857.8 1923.74  4875.9 1915.43  4899.1 1903.08
  4906.8 1897.33  4917.1 1891.13  4927.4 1888.79  4938.2  1888.3    4988 1886.94
  4988.5 1886.44  5005.9 1886.94  5030.3 1887.94  5044.3 1890.23    5074  1890.6
  5133.5 1893.69  5164.5 1895.76  5214.8 1901.35  5253.9  1902.7  5259.5 1903.97
  5304.2 1906.66  5348.9 1913.18  5357.3  1915.2  5410.4 1923.52  5438.4 1926.98
  5446.8 1929.19  5460.7 1929.66  5499.9 1938.26  5522.2 1940.94  5558.6 1943.63
#Mann= 6 ,-1 , 0
  4793.4     .07       0  4938.2      .1       0    4988     .05       0
  5005.9      .1       0    5074    .035       0  5133.5     .07       0
Bank Sta=4988,5005.9
XS Rating Curve= 0 ,0
Exp/Cntr=0.3,0.1

Type RM Length L Ch R = 1 ,6750    ,248,248,248
BEGIN DESCRIPTION:
Fessenden Branch 14.0
END DESCRIPTION:
XS GIS Cut Line= 3
        1859975.     13971175.02        1859975.       13971525.
      1860424.99     13971824.99
#Sta/Elev= 30
  4650.3 1923.52  4670.3 1921.82  4690.3 1918.08  4710.3 1912.63  4730.3 1910.22
    4738 1907.08  4760.3 1900.99  4780.3 1897.08  4850.3 1891.59  4870.3 1891.06
  4895.9 1887.57  4911.3 1886.35  4911.8 1885.85  4929.2 1886.35  5036.3 1886.61
  5049.9 1890.61  5064.9 1891.87  5112.9 1892.29  5144.1 1892.25    5173 1892.26
  5188.1 1894.94  5216.6 1897.19  5245.2 1895.11  5317.3 1898.29  5332.3  1902.5
  5353.3 1905.57  5389.4 1916.02  5432.9 1925.68  5505.1 1937.94  5541.1 1941.46
#Mann= 7 ,-1 , 0
  4650.3      .1       0    4738     .07       0  4895.9      .1       0
  4911.3     .05       0  4929.2      .1       0  5112.9     .07       0
  5144.1      .1       0
Bank Sta=4911.3,4929.2
XS Rating Curve= 0 ,0
Exp/Cntr=0.3,0.1

Type RM Length L Ch R = 1 ,6502    ,166,166,166
BEGIN DESCRIPTION:
Mapping XS 37d3fa8d
END DESCRIPTION:
XS GIS Cut Line= 2
      1859787.55     13971181.28      1859785.53     13972259.87
#Sta/Elev= 30
  4569.1 1922.82  4622.8 1919.23  4642.8 1916.47  4682.8 1909.18  4703.7 1903.78
  4732.8 1895.47  4792.8 1894.02  4822.8 1890.51  4849.4  1889.9  4872.8 1889.43
  4892.8 1887.16  5003.9 1886.65  5004.4 1886.15  5021.8 1886.65  5042.8 1892.21
    5066 1892.73  5112.8 1894.05  5182.8 1891.98  5322.8 1891.05  5342.8 1889.76
  5352.8 1887.45  5382.8 1887.44  5392.8 1888.32  5412.8 1894.64  5442.8 1915.61
  5452.8  1921.7  5457.8  1922.6  5489.5 1927.95  5562.8 1942.42  5647.7  1952.8
#Mann= 8 ,-1 , 0
  4569.1      .1       0  4703.7     .07       0  4849.4      .1       0
  5003.9     .05       0  5021.8      .1       0    5066    .035       0
  5457.8      .1       0  5489.5     .07       0
Bank Sta=5003.9,5021.8
XS Rating Curve= 0 ,0
Exp/Cntr=0.3,0.1

Type RM Length L Ch R = 1 ,6336    ,425,425,425
BEGIN DESCRIPTION:
Fessenden Branch 13.0
END DESCRIPTION:
XS GIS Cut Line= 3
        1859625.     13971225.02        1859625.       13971625.
      1859224.97     13972025.03
#Sta/Elev= 30
  4604.3 1920.66  4624.3 1919.12  4744.3 1904.14  4764.3 1898.79  4774.3 1894.19
  4794.3 1893.93  4804.3 1892.98  4844.3 1887.11  4879.4 1886.93  4955.3  1886.6
  4955.8  1886.1  4973.3  1886.6  5089.1 1892.43  5145.7 1892.91  5173.5 1891.16
  5230.5 1887.43  5326.7 1886.84  5343.7 1886.88    5372 1891.94  5400.3  1905.4
  5414.4 1913.87  5442.7 1938.71  5456.8 1952.05    5471 1960.86  5485.1  1971.2
  5499.3 1977.14  5513.4 1980.76  5531.5 1982.99  5555.8 1984.53    5570 1984.64
#Mann= 7 ,-1 , 0
  4604.3      .1       0  4879.4     .07       0  4955.3     .05       0
  4973.3     .07       0  5173.5      .1       0  5326.7     .07       0
  5531.5      .1       0
Bank Sta=4955.3,4973.3
XS Rating Curve= 0 ,0
Exp/Cntr=0.3,0.1

Type RM Length L Ch R = 1 ,5911    ,447,447,447
BEGIN DESCRIPTION:
Fessenden Branch 12.0
END DESCRIPTION:
XS GIS Cut Line= 3
      1859524.99     13971175.01        1859275.       13971575.
      1859075.02     13971874.97
#Sta/Elev= 30
  4532.4 1922.33  4582.5 1917.51  4597.8 1914.71  4707.5 1902.65  4730.7 1899.09
    4780 1893.23  4877.1 1890.27  4880.9  1889.6  4886.7  1890.2  4896.2 1888.21
  4902.1 1889.86  4909.7 1887.73  4917.4 1887.51  5008.5 1886.73    5009 1886.23
  5026.7 1886.73  5036.7 1886.76    5159 1886.92  5184.4 1886.95  5191.9 1888.57
  5212.9 1896.63  5227.9 1906.43    5249 1917.61    5270 1934.78    5279 1946.37
    5306 1968.95  5315.1 1973.49  5328.6 1982.42  5339.5 1985.69  5364.6 1989.49
#Mann= 8 ,-1 , 0
  4532.4      .1       0  4730.7     .07       0  4877.1     .07       0
  5008.5     .05       0  5026.7     .07       0  5036.7      .1       0
    5159     .07       0  5339.5      .1       0
Bank Sta=5008.5,5026.7
XS Rating Curve= 0 ,0
Exp/Cntr=0.3,0.1

Type RM Length L Ch R = 1 ,5464    ,417,417,417
BEGIN DESCRIPTION:
Fessenden Branch 11.0
END DESCRIPTION:
XS GIS Cut Line= 3
      1859524.97     13971125.02        1859075.       13971425.
        1858725.       13971525.
#Sta/Elev= 30
  4450.9 1923.81    4483 1922.31  4515.5 1919.69  4565.2 1912.94  4638.7 1904.79
  4667.2 1902.69  4731.8 1893.18  4847.5 1891.42    4870 1889.42  4928.6 1888.56
  5008.6 1888.08  5024.2  1886.8  5024.7  1886.3  5042.4  1886.8  5091.5  1887.9
  5159.4 1887.77  5220.5    1889    5227 1897.42  5247.6 1917.33  5260.8 1929.44
    5266 1931.98  5272.5  1946.2  5282.9 1956.36  5293.3 1962.49  5299.8 1971.32
  5304.4 1973.62  5314.1 1980.98  5333.6 1991.65  5345.3 1994.51  5355.7 1995.56
#Mann= 9 ,-1 , 0
  4450.9     .07       0    4483      .1       0  4565.2     .07       0
  4928.6     .07       0  5024.2     .05       0  5042.4     .07       0
  5091.5     .07       0  5247.6      .1       0  5304.4     .07       0
Bank Sta=5024.2,5042.4
XS Rating Curve= 0 ,0
Exp/Cntr=0.3,0.1

Type RM Length L Ch R = 1 ,5047    ,503,503,503
BEGIN DESCRIPTION:
Fessenden Branch 10.0
END DESCRIPTION:
XS GIS Cut Line= 3
        1859475.       13971075.        1859175.       13971075.
      1858724.98       13970975.
#Sta/Elev= 30
    4700 1922.53    4740 1919.02    4790 1911.25    4850 1904.41    4890 1897.73
    4930 1894.21    4940 1892.04    4950 1892.19  4980.9 1886.99  4981.4 1886.49
  4998.6 1886.49  4999.1 1886.99  5174.1 1888.37  5194.6 1887.34  5216.8 1887.25
  5245.9 1887.51  5252.3 1889.06  5257.4 1893.28  5276.6 1905.68  5295.8 1917.86
  5300.9 1920.29  5307.3 1925.72  5338.1 1939.37  5344.5 1943.78    5379 1958.38
  5399.5 1969.45    5420 1977.84    5434 1982.73  5436.6 1983.85    5461  1987.9
#Mann= 5 ,-1 , 0
    4700     .07       0  4980.9     .05       0  4999.1     .07       0
  5216.8      .1       0    5434     .07       0
Bank Sta=4980.9,4999.1
XS Rating Curve= 0 ,0
Exp/Cntr=0.3,0.1

Type RM Length L Ch R = 1 ,4544    ,828,828,828
BEGIN DESCRIPTION:
Fessenden Branch 9.0
END DESCRIPTION:
XS GIS Cut Line= 3
      1859724.49     13970811.16      1859030.95     13970786.82
      1858824.96       13970775.
#Sta/Elev= 30
  4300.5 1925.21  4389.1 1920.83  4410.1 1920.46  4450.1 1915.82  4500.1 1911.53
  4530.1 1907.55  4550.1 1906.01  4650.2 1892.16  4657.1 1891.85  4670.2  1890.8
  4680.2 1888.38  4690.2 1887.29  4920.4 1887.69  4971.3 1886.69  4971.8 1886.19
  4989.5 1886.69  4991.6 1886.81  5020.5 1887.07  5030.5 1896.68  5040.5 1904.49
  5050.5 1911.87  5070.5 1924.71  5100.6 1940.75  5114.5 1946.42  5120.6 1951.14
  5140.7    1961  5150.7 1966.84  5160.7 1970.59    5200 1980.05  5200.8 1980.05
#Mann= 7 ,-1 , 0
  4300.5     .07       0  4389.1      .1       0  4657.1     .07       0
  4971.3     .05       0  4989.5     .07       0  4991.6      .1       0
    5200     .07       0
Bank Sta=4971.3,4989.5
XS Rating Curve= 0 ,0
Exp/Cntr=0.3,0.1

Type RM Length L Ch R = 1 ,3716    ,261,261,261
BEGIN DESCRIPTION:
Fessenden Branch 8.0
END DESCRIPTION:
XS GIS Cut Line= 4
        1860025.       13970075.      1859819.36     13970383.74
        1859475.       13970425.      1858924.95       13970475.
#Sta/Elev= 30
  4282.1 1955.74  4304.6 1954.83  4412.8 1944.35  4454.9 1937.33    4521 1929.22
  4578.1 1919.74  4599.1 1914.36  4606.5 1914.44  4629.2 1911.21  4650.2 1906.49
  4652.5 1904.61  4667.5 1902.33  4697.7 1901.13    4728 1895.91  4745.6 1890.12
  4758.2  1887.3  4768.2 1887.02  4778.3 1887.91  4910.2 1886.61  4910.7 1886.11
  4928.4 1886.61  5322.1 1887.02  5331.2 1887.57  5341.3 1892.84  5361.4 1907.39
  5381.5  1918.2  5431.7 1937.13  5491.9 1950.11    5522 1954.42  5552.2 1956.96
#Mann= 5 ,-1 , 0
  4282.1      .1       0  4745.6     .07       0  4910.2     .05       0
  4928.4     .07       0  5322.1     .07       0
Bank Sta=4910.2,4928.4
XS Rating Curve= 0 ,0
Exp/Cntr=0.3,0.1

Type RM Length L Ch R = 1 ,3455    ,618,618,618
BEGIN DESCRIPTION:
Fessenden Branch 7.1
END DESCRIPTION:
XS GIS Cut Line= 4
      1859944.89     13970141.32      1859738.69     13970273.72
      1859261.26     13970054.54      1859038.92     13970037.27
#Sta/Elev= 30
  4575.4 1944.71  4718.1 1909.42  4825.4 1888.95  4911.3 1883.26  5019.1 1884.92
  5024.6 1879.79  5088.1 1882.52  5093.6 1877.58  5116.5 1884.03    5122 1878.56
  5139.5 1883.18    5145 1877.86  5162.5 1882.21    5168 1876.93  5185.5 1882.82
    5191 1877.19  5208.5 1882.03  5227.8 1874.47  5228.3 1873.97  5246.2 1874.47
    5260 1881.99  5265.5 1875.93    5283 1881.08  5288.5 1875.19  5314.6  1877.8
  5382.2 1904.61  5432.3 1906.84  5483.1 1917.26  5530.6 1921.34  5568.8 1916.77
#Mann= 8 ,-1 , 0
  4575.4      .1       0  4718.1     .07       0  4825.4      .1       0
  4911.3     .07       0  5227.8     .05       0  5246.2     .07       0
  5314.6      .1       0  5483.1     .07       0
Bank Sta=5227.8,5246.2
XS Rating Curve= 0 ,0
Exp/Cntr=0.3,0.1

Type RM Length L Ch R = 1 ,2837    ,445,445,445
BEGIN DESCRIPTION:
Fessenden Branch 6.0
END DESCRIPTION:
XS GIS Cut Line= 3
        1860075.       13969625.        1859475.       13969775.
      1859174.97     13969925.01
#Sta/Elev= 30
  4389.6 1987.31  4412.8 1983.57    4454 1966.88  4482.4 1950.76  4490.1 1944.49
  4495.2 1944.26  4531.3 1921.26  4536.5  1920.8  4572.6 1896.95  4577.7 1897.34
  4585.4 1891.83  4606.2 1882.58  4626.7 1876.44  4667.9  1870.8  4783.9  1869.3
  4840.7  1864.3  4915.2 1862.71  4925.6 1860.39  4975.7 1859.25  4976.2 1858.75
  4994.1 1859.25  4997.8 1859.34  5005.5 1864.34  5066.8 1867.29  5075.8 1869.65
  5178.6 1876.78  5245.6 1886.48  5262.4 1891.81  5307.1  1900.5  5343.5 1901.56
#Mann= 7 ,-1 , 0
  4389.6      .1       0  4606.2     .07       0  4840.7      .1       0
  4915.2     .07       0  4975.7     .05       0  4994.1     .07       0
  5075.8      .1       0
Bank Sta=4975.7,4994.1
XS Rating Curve= 0 ,0
Exp/Cntr=0.3,0.1

Type RM Length L Ch R = 1 ,2392    ,375,375,375
BEGIN DESCRIPTION:
Fessenden Branch 5.0
END DESCRIPTION:
XS GIS Cut Line= 3
      1860075.05       13969425.        1859725.       13969425.
      1859125.02       13969525.
#Sta/Elev= 30
  4650.4 1993.64  4652.9 1993.64  4690.4 1981.79  4730.4  1960.2  4820.4  1907.1
  4850.4  1892.2  4870.4 1884.28  4913.5 1870.38  4961.2 1857.12  4961.7 1856.62
  4979.6 1857.12  5046.5 1857.85    5112 1861.61  5122.1 1864.87  5132.2 1866.88
    5150 1868.54  5155.8 1867.93  5182.9 1869.37  5276.7 1869.64  5337.5 1871.34
  5448.6 1881.36  5459.2 1882.78  5466.8  1885.3  5507.3 1891.94  5514.9 1894.19
    5520 1894.12  5575.8  1905.6  5580.8 1904.78  5588.4 1907.11  5608.7 1908.52
#Mann= 7 ,-1 , 0
  4650.4      .1       0  4913.5     .07       0  4961.2     .05       0
  4979.6     .07       0  5046.5      .1       0  5155.8     .07       0
  5448.6      .1       0
Bank Sta=4961.2,4979.6
XS Rating Curve= 0 ,0
Exp/Cntr=0.3,0.1

Type RM Length L Ch R = 1 ,2017    ,91,91,91
BEGIN DESCRIPTION:
Fessenden Branch 4.1
END DESCRIPTION:
XS GIS Cut Line= 5
      1859955.67     13969006.36      1859732.18     13969006.36
      1859706.14     13969017.21      1859673.59      13969069.3
      1859404.52      13969249.4
#Sta/Elev= 30
  4689.8 1979.41  4692.6 1979.41  4720.5 1967.14  4730.5 1963.55  4780.5 1948.46
  4853.1 1919.09  4880.5 1907.54  4890.5 1899.49  4900.5 1885.81  4909.4 1877.95
  4913.3 1877.95  4919.2 1866.97  4924.6 1862.31  4939.4 1847.61  4943.5  1847.5
  4945.6 1847.38  4946.1 1846.88  4964.1 1847.38  4966.9 1847.78  4985.5 1848.63
  4991.4 1847.84  5005.7 1850.03  5020.7 1848.94  5035.7 1853.14  5056.7 1863.68
  5071.8 1865.02  5092.8 1866.52  5223.2 1868.64  5293.9 1867.93  5326.7 1869.35
#Mann= 7 ,-1 , 0
  4689.8      .1       0  4853.1    .035       0  4943.5     .07       0
  4945.6     .05       0  4964.1     .07       0  4966.9    .035       0
  5223.2      .1       0
Bank Sta=4945.6,4964.1
XS Rating Curve= 0 ,0
Exp/Cntr=0.3,0.1
