HEC-RAS study Guadalupe River.prj: Guadalupe River Base Level Engineering

--- Guadalupe River.g01 (geometry) --- (continued)

Type RM Length L Ch R = 1 ,2328253 ,1409,1409,1409
BEGIN DESCRIPTION:
Guadalupe River - 217
END DESCRIPTION:
XS GIS Cut Line= 4
      1827486.26     13935743.85      1827600.19     13934984.34
      1828283.79      13933908.3      1829043.31     13933528.54
#Sta/Elev= 30
  3952.9  2085.4  4115.8 2079.32  4179.8  2066.7  4333.6 2049.97  4370.1 2043.67
  4455.6 2033.13  4548.3 2016.49  4648.3 1985.99  4653.4 1987.07    4667 1980.26
  4717.4 1965.18  4744.5 1965.44  4759.7 1959.88    4775    1940  4832.6 1891.98
  4838.6  1869.3  4847.8 1859.17  4853.7 1861.58  4862.3 1855.66  4952.4 1853.01
  5028.2 1857.24  5128.8 1869.67  5239.1 1874.14  5302.6  1882.5  5426.3 1888.81
  5608.7 1899.68  5954.8 1939.33  6146.7 1946.59  6210.6 1948.25  6844.9 1969.36
#Mann= 11 ,-1 , 0
  3952.9     .07       0  4333.6     .05       0  4370.1     .07       0
  4455.6     .05       0    4667     .12       0  4862.3     .04       0
  5028.2     .05       0  5128.8     .12       0  5426.3     .07       0
  6146.7     .12       0  6210.6     .07       0
Bank Sta=4862.3,5028.2
XS Rating Curve= 0 ,0
Exp/Cntr=0.3,0.1

Type RM Length L Ch R = 1 ,2326844 ,1504,1504,1504
BEGIN DESCRIPTION:
Guadalupe River - 216
END DESCRIPTION:
XS GIS Cut Line= 3
      1828271.13     13935883.14      1828891.43     13935300.82
      1829347.16     13933515.89
#Sta/Elev= 30
  3967.7 2028.93  4103.5 2017.46  4195.4 2015.08  4414.7 1995.34  4619.8 1967.83
  4683.8 1955.08  4733.1 1951.17  4817.5 1932.76  4851.7 1932.31  4856.9 1929.48
  4907.1 1924.75  4917.4 1917.02  4927.7    1905  4933.4 1891.45  4938.6 1894.77
  4944.1 1870.63  4948.4 1851.76  5021.7 1849.45  5132.5 1853.03  5178.6  1854.7
  5246.2 1872.33  5319.9 1877.54  5517.4 1878.83  5608.9 1881.29  5622.8 1881.72
  5658.5 1891.57  5903.6 1938.12  6109.5 1952.78  6184.4 1958.52  6660.7 1976.73
#Mann= 8 ,-1 , 0
  3967.7     .12       0  4944.1     .07       0  4948.4     .04       0
  5132.5     .07       0  5246.2     .12       0  5517.4     .07       0
  5608.9     .12       0  6109.5     .07       0
Bank Sta=4948.4,5132.5
XS Rating Curve= 0 ,0
Exp/Cntr=0.3,0.1

Type RM Length L Ch R = 1 ,2325340 ,1524,1524,1524
BEGIN DESCRIPTION:
Guadalupe River - 215
END DESCRIPTION:
XS GIS Cut Line= 2
      1830372.57     13935845.21      1829879.07     13933478.92
#Sta/Elev= 30
  4194.9 2036.24    4309 2047.39    4404 2049.23    4504 2034.83    4699 1975.59
  4716.1 1963.54  4787.6 1938.69  4862.3 1904.08    4894  1893.9  4910.2 1882.65
  4920.4 1865.18  4930.6 1859.71  4961.2 1852.37  4990.1 1849.59    5089 1851.52
  5194.7 1854.88  5257.5 1864.88  5348.6 1869.85  5666.1 1874.44  5696.7 1882.92
    5727 1906.19  5737.6 1912.64    5758  1915.5  5774.1 1926.61    5819 1943.68
  5919.1 1953.82  6045.5 1959.29  6196.7 1971.24  6316.3 1978.39  6612.1 1992.25
#Mann= 10 ,-1 , 0
  4194.9     .07       0  4862.3     .12       0  4961.2     .04       0
    5089     .12       0  5194.7     .12       0  5348.6     .07       0
    5727     .12       0  6045.5     .07       0  6196.7     .05       0
  6316.3     .07       0
Bank Sta=4961.2,5089
XS Rating Curve= 0 ,0
Exp/Cntr=0.3,0.1

Type RM Length L Ch R = 1 ,2323816 ,1508,1508,1508
BEGIN DESCRIPTION:
Guadalupe River - 214
END DESCRIPTION:
XS GIS Cut Line= 2
      1832018.28     13935414.77      1830271.27     13933123.39
#Sta/Elev= 30
  3977.1  2060.6  4077.5 2057.66  4350.7 2051.75  4421.4 2027.46  4507.6 1977.49
  4541.9 1958.28  4633.4 1901.07  4699.9 1865.32  4799.7 1861.49  4843.3  1849.4
  4884.9  1850.3  4952.7 1848.01  5028.3 1852.61  5234.3 1864.94  5348.5 1863.41
  5419.9 1854.94  5462.8 1854.46  5477.3 1857.66  5485.6 1864.74  5491.9 1859.01
  5506.4  1900.2  5512.7 1898.78  5520.9 1909.06  5570.8  1926.2  5620.7 1936.68
  5776.7 1942.92  6254.8 1976.35    6670 1991.29  6681.5 1991.43  6858.5 1996.85
#Mann= 10 ,-1 , 0
  3977.1     .07       0  4077.5     .12       0  4507.6     .07       0
  4541.9     .12       0  4633.4     .07       0  4884.9    .035       0
  5028.3     .07       0  5419.9     .12       0    6670     .05       0
  6681.5     .07       0
Bank Sta=4884.9,5028.3
XS Rating Curve= 0 ,0
Exp/Cntr=0.3,0.1

Type RM Length L Ch R = 1 ,2322308 ,1424,1424,1424
BEGIN DESCRIPTION:
Guadalupe River - 213
END DESCRIPTION:
XS GIS Cut Line= 3
      1833220.88     13934389.34      1831815.72     13933465.23
      1830588.84     13933224.91
#Sta/Elev= 30
  3729.1 2015.34  3852.6 2020.59  3945.9 2018.01  4011.2 2011.24  4126.7 1991.46
  4168.8 1978.12  4235.2 1978.04  4286.4 1969.89  4322.5 1955.06  4394.4 1912.41
  4415.9  1893.8    4437 1881.91  4452.1 1854.04  4458.1 1849.87  4552.5 1853.08
  4617.7 1858.19  4700.6  1855.9  4940.4 1853.58    4957 1852.35  4986.5 1847.52
  5117.4 1846.52  5136.5 1848.63  5150.9 1874.77  5181.1 1888.85  5280.5 1912.37
  5388.9 1929.66    6220 1965.41  6399.1 1972.79  6400.7 1972.85  6661.1 1983.61
#Mann= 10 ,-1 , 0
  3729.1     .07       0  4011.2     .12       0  4552.5     .07       0
  4700.6     .12       0  4940.4     .05       0    4957    .035       0
  5136.5     .05       0    6220     .07       0  6399.1     .05       0
  6400.7     .07       0
Bank Sta=4957,5136.5
XS Rating Curve= 0 ,0
Exp/Cntr=0.3,0.1

Type RM Length L Ch R = 1 ,2320884 ,1150,1150,1150
BEGIN DESCRIPTION:
Guadalupe River - 212
END DESCRIPTION:
XS GIS Cut Line= 4
      1834005.76     13933275.33      1832701.87     13932553.76
      1832005.61     13932781.63      1830651.07     13932705.67
#Sta/Elev= 30
  3837.3 1975.83  4117.5 1963.86  4375.3 1935.69  4426.7 1925.87  4486.2 1905.26
  4523.9 1887.16  4535.5 1857.69  4558.2 1848.74  4584.4 1847.08  4727.8 1853.13
  4733.7 1853.19  4860.7    1853  4913.3 1847.73  4969.7 1844.07  4982.1 1840.35
  5045.1 1842.09  5134.6 1843.76  5286.3 1870.66  5343.8 1891.72  5524.2 1921.94
  5738.3 1934.52  6051.1 1937.12  6411.3 1934.53  6609.4 1939.61    6642 1941.45
  6819.9 1947.83  6826.1  1948.2  7164.4 1966.07  7174.1 1965.79  7416.8  1974.4
#Mann= 17 ,-1 , 0
  3837.3     .12       0  4584.4     .07       0  4727.8     .12       0
  4733.7     .07       0  4913.3     .12       0  4969.7     .04       0
  5045.1     .12       0  5134.6     .12       0  5286.3     .07       0
  5738.3     .12       0  6051.1     .07       0  6609.4     .12       0
    6642     .07       0  6819.9     .12       0  6826.1     .07       0
  7164.4     .12       0  7174.1     .07       0
Bank Sta=4969.7,5045.1
XS Rating Curve= 0 ,0
Exp/Cntr=0.3,0.1

Type RM Length L Ch R = 1 ,2319734 ,767,767,767
XS GIS Cut Line= 5
  1834204.48367913933090.1251309 1833453.615430513932413.0418394
  1833592.05806713932242.2298451 1833981.466408913931833.3510696
  1833695.90037913931086.9857645
#Sta/Elev= 30
       0 1963.08  267.63 1961.32  465.88 1945.99     565 1934.88   644.3 1916.72
  703.78 1896.24   723.6 1888.71  743.43 1859.06  753.34 1852.42  773.16 1848.94
  862.38 1847.29  921.85 1842.44  941.68 1843.06  981.33  1852.4 1160.97 1850.76
 1448.86 1842.68 1478.58 1839.59  1508.3 1836.04 1577.64    1838 1726.23 1839.13
 1805.56 1842.93 1965.39 1841.73 2015.33 1848.32 2115.23  1852.9 2145.19 1859.28
 2384.93 1858.98 2404.91 1865.38 2444.87 1887.74  2504.8  1933.6 2594.71 1977.08
#Mann= 4 ,-1 , 0
       0     .12       0  703.78     .06       0 1478.58     .04       0
 1577.64      .1       0
Bank Sta=1478.58,1577.64
XS Rating Curve= 0 ,0
Exp/Cntr=0.3,0.1

Type RM Length L Ch R = 1 ,2318967 ,2486,2486,2486
BEGIN DESCRIPTION:
Guadalupe River - 211
END DESCRIPTION:
XS GIS Cut Line= 3
      1834143.26     13933561.53      1834512.18     13932454.75
      1834251.81     13930089.69
#Sta/Elev= 30
    3274 1969.07  3597.1    1968  4296.4 1932.36  4486.5 1927.89  4585.8 1925.49
  4685.1 1918.01  4782.4 1906.02  4883.1 1880.09  4912.8 1867.35  4917.9 1844.04
  4923.3 1835.95  4945.5  1828.8  5029.6  1829.8    5044 1836.15  5065.6 1839.24
  5325.7 1846.33  5446.4 1837.76  5496.7 1853.36  5777.5 1854.79  5848.9 1855.98
  5889.1 1863.39  5923.5 1880.67  5969.6 1912.85  6019.9 1960.98    6040 1971.92
  6105.4 2002.85    6211 2042.62  6317.8 2066.46  6527.3 2066.89    6820 2071.85
#Mann= 11 ,-1 , 0
    3274     .12       0  4296.4     .07       0  4486.5     .12       0
  4585.8     .07       0  4685.1     .12       0  4923.3     .04       0
    5044     .12       0  5065.6     .07       0  5777.5     .12       0
  6317.8     .07       0  6527.3     .12       0
Bank Sta=4923.3,5044
XS Rating Curve= 0 ,0
Exp/Cntr=0.3,0.1

Type RM Length L Ch R = 1 ,2316481 ,1438,1438,1438
BEGIN DESCRIPTION:
Guadalupe River - 210
END DESCRIPTION:
XS GIS Cut Line= 4
      1834425.39     13934169.15       1836400.2     13932758.57
      1836660.62     13932020.72      1835380.25     13930783.75
#Sta/Elev= 30
  2206.5 1957.36  2313.1 1952.53  2355.7 1950.26  2420.9 1946.79  2926.3 1921.43
  3004.8 1912.16    3134 1916.89  3442.4 1909.01  3599.7 1890.04  3958.6 1869.15
  4029.8  1872.9  4331.3 1861.72  4435.5 1857.92  4510.3 1855.19  4923.5 1843.02
  4944.7 1837.27  4976.5 1834.73  4995.6 1827.72    5116 1826.72  5158.6 1827.72
  5178.4 1833.99  5188.6  1852.1  5198.8 1903.79  5260.6 1921.25  5414.9 1929.18
  5862.3 1967.14  6300.7 1982.43  6703.8 2029.07  6930.2 2032.09  7196.1 2019.67
#Mann= 9 ,-1 , 0
  2206.5     .07       0  2313.1     .08       0  2355.7     .07       0
  2420.9     .12       0  4331.3     .05       0  4435.5     .12       0
  4510.3     .07       0  4923.5     .04       0  5178.4     .12       0
Bank Sta=4923.5,5178.4
XS Rating Curve= 0 ,0
Exp/Cntr=0.3,0.1

Type RM Length L Ch R = 1 ,2315043 ,1247,1247,1247
XS GIS Cut Line= 4
  1835681.78026513933941.2313683 1837469.974523713933403.0369066
 1837834.558112113932856.1620161 1837999.4885566 13932222.481525
#Sta/Elev= 30
       0 1922.69   219.7 1906.78  459.37 1882.79   509.3 1880.06  539.26 1879.25
  589.19    1868  758.96 1856.03  878.79 1851.99 1687.68 1846.73 1937.14 1842.62
 1957.06 1843.12 1976.97 1840.72 1996.89 1842.12 2016.81 1831.75 2026.77 1830.39
 2116.39  1827.3 2166.18 1830.19 2235.89 1830.06 2335.48  1838.8 2464.94 1843.74
 2663.58 1846.72 2703.27 1845.48 2742.95 1836.11 2792.56 1840.24 2832.24 1841.06
 2852.08  1848.1 2941.37 1888.93 3010.82 1907.37 3149.71  1949.1 3179.48 1954.64
#Mann= 6 ,-1 , 0
       0     .11       0   509.3     .05       0 1937.14     .12       0
 2026.77     .04       0 2166.18     .06       0 2663.58     .12       0
Bank Sta=2026.77,2166.18
XS Rating Curve= 0 ,0
Exp/Cntr=0.3,0.1

Type RM Length L Ch R = 1 ,2313796 ,2662,2662,2662
BEGIN DESCRIPTION:
Guadalupe River - 209
END DESCRIPTION:
XS GIS Cut Line= 4
      1839134.59     13934993.83      1838548.64     13934104.06
      1838570.34     13932736.87      1839156.28     13931695.19
#Sta/Elev= 30
  3456.4 2021.92  3694.4 1990.86  3798.7 1980.31  3833.1 1976.81    4011 1949.66
  4227.8 1922.99  4620.8 1886.68  4630.8 1883.43  4640.8 1869.33  4670.8 1841.64
  4680.8  1837.2  4730.9 1834.16  4890.9 1837.66  4940.9 1825.41  4967.2 1823.81
  5040.9 1825.31  5303.4 1833.97  5430.9 1830.78    5531 1841.17  5635.5 1843.98
    6098 1849.12  6135.6 1858.77  6151.1 1868.66  6157.3 1868.64  6173.2 1879.08
  6210.8  1888.9  6459.4 1942.97  6658.9 1974.13  6826.5 1993.27  7084.3 2006.36
#Mann= 9 ,-1 , 0
  3456.4     .12       0  3694.4     .07       0  3798.7     .12       0
  3833.1     .07       0  4940.9     .04       0  5040.9     .07       0
  5303.4     .12       0  5635.5     .07       0  6151.1     .12       0
Bank Sta=4940.9,5040.9
XS Rating Curve= 0 ,0
Exp/Cntr=0.3,0.1

Type RM Length L Ch R = 1 ,2311134 ,1473,1473,1473
BEGIN DESCRIPTION:
Guadalupe River - 208
END DESCRIPTION:
XS GIS Cut Line= 2
      1840715.18     13934604.55      1840474.65     13932275.23
#Sta/Elev= 30
  3796.3 1972.19  3956.7 1939.82  4320.3 1896.16  4333.6 1893.69  4338.7  1886.2
  4348.8 1859.56  4358.8 1851.77    4399 1829.48  4419.1 1824.19  4469.4 1822.46
  4526.5 1828.18  4666.2 1831.38  4830.2  1825.1  4901.7 1818.02  4982.1 1817.86
  5021.3 1813.34  5052.5 1819.09  5098.1 1822.68  5273.7 1820.84  5302.9 1827.77
    5308 1824.57    5344 1835.49  5756.2 1834.21  5808.5    1839  5886.6 1891.01
  5891.2 1890.53  5917.1 1920.09  5927.1 1924.99  6007.5 1945.88    6138 1955.42
#Mann= 8 ,-1 , 0
  3796.3     .12       0  4320.3     .07       0  4666.2     .12       0
  4830.2     .07       0  4982.1     .04       0  5052.5     .07       0
  5098.1     .07       0  5808.5     .12       0
Bank Sta=4982.1,5052.5
XS Rating Curve= 0 ,0
Exp/Cntr=0.3,0.1

Type RM Length L Ch R = 1 ,2309661 ,1129,1129,1129
BEGIN DESCRIPTION:
Guadalupe River - 207
END DESCRIPTION:
XS GIS Cut Line= 2
      1841867.18      13934515.9      1841955.79     13931971.44
#Sta/Elev= 30
  4238.5 1927.54  4279.4 1922.16  4369.5 1915.46  4439.5 1905.35  4689.7 1879.18
  4719.7 1871.22  4759.7 1864.33  4789.7 1851.54  4809.7 1847.76  4829.8 1837.63
  4839.8 1829.82  4859.8 1822.11  4879.8 1817.52  4899.8 1816.45  4909.8 1813.67
  4956.3 1812.47  5069.9  1814.6  5089.9 1817.55  5109.9 1824.42  5129.9 1827.33
  5221.8 1832.05  5370.1  1833.6  5630.2 1827.66  6044.5 1834.18  6150.6 1838.52
  6182.7 1849.66  6390.7 1921.42  6480.8 1949.26  6610.8 1978.48  6784.5  2000.2
#Mann= 5 ,-1 , 0
  4238.5     .12       0  4899.8    .035       0  5069.9     .12       0
  5221.8     .07       0  6182.7     .12       0
Bank Sta=4899.8,5069.9
XS Rating Curve= 0 ,0
Exp/Cntr=0.3,0.1

Type RM Length L Ch R = 1 ,2308532 ,1478,1478,1478
BEGIN DESCRIPTION:
Guadalupe River - 206
END DESCRIPTION:
XS GIS Cut Line= 4
      1843004.92     13934949.04      1842972.98     13934052.35
      1842746.41     13933417.81      1842772.81     13932048.19
#Sta/Elev= 30
  3648.1 1931.15  3932.3 1910.65  4092.4 1889.87  4252.5 1862.48  4344.6 1855.59
  4472.7  1850.6  4512.7  1846.7  4574.4    1833  4699.7 1828.49  4795.8 1819.75
  4923.6 1813.62  4925.1 1812.42  5019.6 1813.62  5064.6 1814.87  5105.3 1819.63
  5171.5 1817.81    5332 1827.52    5452 1824.22    5482 1815.67    5522 1826.18
    5552 1828.22  5882.1 1831.46  5972.1 1837.77  6039.5 1863.87  6072.1 1872.19
  6112.1 1874.54  6202.1 1856.34  6232.1 1855.96  6342.1 1891.36    6589 1949.23
#Mann= 8 ,-1 , 0
  3648.1     .12       0  4344.6     .07       0  4795.8     .12       0
  4923.6     .05       0  5019.6     .12       0  5064.6     .12       0
  5171.5     .07       0  6039.5     .12       0
Bank Sta=4923.6,5019.6
XS Rating Curve= 0 ,0
Exp/Cntr=0.3,0.1

Type RM Length L Ch R = 1 ,2307054 ,1282,1282,1282
BEGIN DESCRIPTION:
Guadalupe River - 205
END DESCRIPTION:
XS GIS Cut Line= 2
       1843044.5     13935047.61      1844196.21     13932769.49
#Sta/Elev= 30
  3062.4 1934.44  3222.2 1929.51  3339.3 1918.47  3407.1  1914.8    3523 1898.87
  3715.5 1866.78  3823.9  1852.8  3999.9 1831.31  4040.8 1825.01  4162.2 1828.24
  4233.4 1827.58  4261.3 1827.36  4704.1 1821.03    4917 1818.92  4970.2 1808.22
  4985.2 1803.14  5044.5 1804.34  5082.3 1809.91  5104.7 1822.94    5112  1831.5
  5117.6 1846.93  5127.1 1885.45  5139.9 1896.83  5149.5 1901.46  5162.2 1914.57
  5223.4 1948.74  5312.6 1977.36  5379.4 1990.28  5468.6 2004.18  5615.1 2021.18
#Mann= 13 ,-1 , 0
  3062.4     .12       0  3339.3     .07       0    3523     .12       0
  3715.5     .07       0  3823.9     .05       0  3999.9     .07       0
  4040.8     .05       0  4162.2     .07       0  4233.4     .05       0
  4261.3     .07       0  4704.1     .05       0  4970.2     .04       0
  5044.5     .12       0
Bank Sta=4970.2,5044.5
XS Rating Curve= 0 ,0
Exp/Cntr=0.3,0.1

Type RM Length L Ch R = 1 ,2305772 ,1260,1260,1260
BEGIN DESCRIPTION:
Guadalupe River - 204
END DESCRIPTION:
XS GIS Cut Line= 3
      1844272.43     13935554.01      1844348.39     13934971.68
       1845209.2      13933515.9
#Sta/Elev= 30
    3155 1920.23  3216.5 1918.68  3527.5 1894.47  3601.4  1884.3  3744.8 1847.76
  3857.9 1836.88  3904.7 1829.48  4154.4 1824.44  4234.4 1817.34  4330.2 1818.27
  4359.5  1818.2    4447 1822.85  4702.5 1824.54  4745.4 1822.42  4844.3 1807.78
  4883.8 1803.31  4942.4 1803.59  4959.4 1801.16  5016.3 1804.61  5051.2 1820.64
  5074.4 1839.12  5080.8 1866.93  5086.6 1879.66  5102.3 1902.07  5139.3 1925.37
  5182.2 1943.73  5225.4 1967.87  5277.8 1985.96  5314.9 1991.38  5433.5 1991.21
#Mann= 7 ,-1 , 0
    3155     .12       0  3857.9     .07       0  4330.2     .12       0
  4359.5     .07       0  4844.3     .12       0  4942.4     .04       0
  5016.3     .12       0
Bank Sta=4942.4,5016.3
XS Rating Curve= 0 ,0
Exp/Cntr=0.3,0.1

Type RM Length L Ch R = 1 ,2304512 ,1116,1116,1116
BEGIN DESCRIPTION:
Guadalupe River - 203
END DESCRIPTION:
XS GIS Cut Line= 2
      1845044.68     13935921.08      1846120.35     13934275.93
#Sta/Elev= 30
  3463.8 1906.01  3671.4 1891.59  3749.7 1878.85    3780 1869.56  3829.5 1862.68
  3851.6 1855.94  3901.2 1832.55  3930.7 1826.75  4211.7 1819.89    4432 1815.79
  4624.4 1822.29  4696.8 1821.49  4752.1 1816.44  4784.3 1807.09    4869 1801.92
  4940.2 1801.91    4944 1801.81  4945.5 1800.61    5017 1801.81  5022.5 1805.87
  5058.7 1813.78  5077.6 1824.48    5116 1851.74    5122 1862.14  5137.1 1876.31
  5275.2 1943.99    5297 1958.04  5354.3 1982.39  5390.5 1988.88  5429.4 1990.07
#Mann= 9 ,-1 , 0
  3463.8     .12       0  3851.6     .07       0  4211.7     .12       0
    4432     .07       0  4752.1     .12       0  4940.2    .035       0
    4944     .04       0  5022.5    .035       0  5077.6     .12       0
Bank Sta=4944,5022.5
XS Rating Curve= 0 ,0
Exp/Cntr=0.3,0.1

Type RM Length L Ch R = 1 ,2303396 ,807,807,807
BEGIN DESCRIPTION:
Guadalupe River - 202
END DESCRIPTION:
XS GIS Cut Line= 2
      1846032.06     13936465.49      1846904.78     13934568.29
#Sta/Elev= 30
    3580 1928.11  3787.3 1904.21  3840.9 1903.99  3953.6  1898.2  3965.8 1890.48
  4010.6  1885.5    4074 1849.23  4079.5 1852.75  4096.9 1844.21  4102.3  1846.9
  4125.4 1834.79  4217.3 1810.77    4269    1809  4375.7  1810.2  4482.4 1812.74
    4589 1811.44  4732.7 1806.79  4881.6 1804.55  4956.4 1803.82  5018.8 1796.34
  5044.5 1804.86  5054.3 1816.01  5066.5 1820.12  5200.1 1821.59  5229.1 1823.02
  5300.6 1836.65  5461.4 1909.76  5512.8 1928.28  5581.7 1943.71  5668.3 1952.31
#Mann= 13 ,-1 , 0
    3580     .12       0  3840.9     .07       0  4102.3     .12       0
    4269     .07       0  4375.7     .12       0  4482.4     .05       0
    4589     .07       0  4732.7     .12       0  4881.6     .07       0
  4956.4     .04       0  5044.5     .07       0  5200.1     .05       0
  5229.1     .12       0
Bank Sta=4956.4,5044.5
XS Rating Curve= 0 ,0
Exp/Cntr=0.3,0.1

Type RM Length L Ch R = 1 ,2302589 ,1100,1100,1100
XS GIS Cut Line= 4
  1846704.49772113936547.6116542 1846871.016417113935850.9535987
 1847383.169264213935677.3423974 1847417.891307613934791.9258612
#Sta/Elev= 30
       0 1932.39   69.64 1918.53  179.07 1900.82  238.76 1884.63  387.99 1862.56
  397.93 1859.43  417.83 1841.62  457.62 1815.29  467.57 1810.52  487.47 1805.79
  517.32 1804.42  716.28 1810.14  794.94 1807.94   844.1 1804.99  863.77 1802.07
  883.43 1797.14  912.93  1795.1 1001.42 1794.31 1050.58 1796.78 1158.74 1812.93
 1257.06 1815.36 1605.53 1819.41 1734.96 1817.36 1834.52 1817.94  1884.3 1820.52
 1904.21 1823.62 1934.08 1834.21 2093.38 1905.28 2103.34 1908.09 2143.16 1913.55
#Mann= 6 ,-1 , 0
       0     .12       0  487.47     .05       0  863.77      .1       0
  883.43     .04       0 1050.58     .09       0 1257.06     .05       0
Bank Sta=883.43,1050.58
XS Rating Curve= 0 ,0
Exp/Cntr=0.3,0.1

Type RM Length L Ch R = 1 ,2301489 ,1953,1953,1953
BEGIN DESCRIPTION:
Guadalupe River - 201
END DESCRIPTION:
XS GIS Cut Line= 4
      1847302.68     13937039.91      1847935.26     13936428.41
      1847766.57     13934783.62      1847049.82     13934678.22
#Sta/Elev= 30
  4102.7 1943.21    4136 1941.41  4284.7 1913.49  4404.8 1899.55  4645.4 1853.34
  4864.5  1835.7  4935.3 1823.77  4942.2 1820.02  4951.3 1821.62  4963.6 1820.57
  4970.5 1807.58  4977.7 1805.52  4981.4 1799.71  4986.8 1799.71  4990.4 1792.68
  5026.5 1791.48  5056.3 1794.47  5116.6 1797.97  5237.3 1796.15  5342.8  1802.2
  5404.3  1812.2  5618.2 1818.94  6033.5 1818.63  6175.8  1817.7  6414.8 1817.61
  6443.6 1819.83  6484.7 1834.82  6564.2 1875.37  6632.7 1902.09  7360.4 1938.58
#Mann= 10 ,-1 , 0
  4102.7     .07       0  4951.3     .12       0  4986.8     .04       0
  5056.3     .12       0  5342.8     .12       0  5404.3     .07       0
  6033.5     .05       0  6175.8     .07       0  6414.8     .05       0
  6484.7     .12       0
Bank Sta=4986.8,5056.3
XS Rating Curve= 0 ,0
Exp/Cntr=0.3,0.1

Type RM Length L Ch R = 1 ,2299536 ,1840,1840,1840
BEGIN DESCRIPTION:
Guadalupe River - 200
END DESCRIPTION:
XS GIS Cut Line= 3
      1850128.31     13936154.28      1848230.48     13934699.27
      1847112.87     13934636.01
#Sta/Elev= 30
  4156.3 2028.31  4358.2 2010.76  4654.4 1955.04  4665.4 1951.82  4721.7 1930.06
    4728 1883.82  4736.2 1862.68  4765.2 1840.39  4821.4 1810.05  4842.2 1792.25
  4907.8 1788.19  4914.8 1788.22  4945.1 1786.49  5020.8 1791.05  5056.1 1791.34
  5099.7 1806.24  5160.6 1807.09  5389.2 1811.24  5393.8 1811.31  5756.4 1814.53
  5857.9  1814.4  6051.8 1814.61  6351.5 1817.19  6412.4 1819.53  6526.6 1864.13
  6603.3  1881.6  6763.5 1897.82    7034 1907.48  7194.2 1918.65  7667.1 1939.84
#Mann= 13 ,-1 , 0
  4156.3     .12       0  4654.4     .07       0  4665.4     .12       0
  4907.8    .035       0  4914.8     .04       0  5020.8     .12       0
  5160.6     .05       0  5389.2     .12       0  5393.8     .05       0
  5756.4     .07       0  5857.9     .05       0  6051.8     .07       0
  6351.5     .12       0
Bank Sta=4914.8,5020.8
XS Rating Curve= 0 ,0
Exp/Cntr=0.3,0.1

Type RM Length L Ch R = 1 ,2297696 ,1926,1926,1926
BEGIN DESCRIPTION:
Guadalupe River - 199
END DESCRIPTION:
XS GIS Cut Line= 2
      1851203.76     13935437.34      1850023.46     13933118.89
#Sta/Elev= 30
  4039.6 1940.78  4120.8 1930.03  4220.4 1923.86    4412 1897.64  4491.5 1884.52
  4569.6 1868.82  4642.8 1844.35  4726.2 1825.41  4808.8 1812.58  4827.8 1808.56
  4931.9 1802.62  4948.6 1799.24  4962.4 1788.87  5003.3 1784.33  5029.7 1787.74
  5084.2 1791.09    5533 1800.37  5723.9 1798.62  5848.9 1792.28  5893.7 1803.94
  5963.6 1802.22  6010.6 1806.77  6055.1  1820.7  6166.3 1883.11    6233 1930.43
  6249.6 1961.83  6318.5 1971.98  6445.9 1969.45  6538.8 1963.36  6641.2 1964.33
#Mann= 14 ,-1 , 0
  4039.6     .07       0  4220.4     .12       0    4412     .07       0
  4491.5     .12       0  4808.8     .07       0  4827.8     .12       0
  4962.4     .04       0  5029.7     .12       0  5084.2     .07       0
    5533     .05       0  5723.9     .07       0  5963.6     .12       0
  6318.5     .07       0  6445.9     .12       0
Bank Sta=4962.4,5029.7
XS Rating Curve= 0 ,0
Exp/Cntr=0.3,0.1

Type RM Length L Ch R = 1 ,2295770 ,1868,1868,1868
BEGIN DESCRIPTION:
Guadalupe River - 198
END DESCRIPTION:
XS GIS Cut Line= 3
      1851752.03     13935352.94      1852110.49     13934741.45
      1851625.49     13932274.28
#Sta/Elev= 30
    2671 1927.36  2856.6 1921.73  2945.5 1916.75  3102.7 1909.44  3262.9 1894.16
  3386.9 1869.21  3435.2 1850.11  3489.7 1828.72  3498.5 1817.75  3529.1 1819.14
  3565.6 1806.49  3877.9 1804.34  4079.6 1803.75  4204.6 1803.51  4514.7 1801.47
  4741.8 1797.86  4831.2 1785.61  4939.1 1785.24  4964.6 1779.86  5027.2 1786.16
  5189.2 1782.83  5201.2 1795.27    5231 1805.65  5271.8 1833.29  5298.9  1872.5
  5350.3 1909.36  5401.7 1925.78  5453.1 1937.89  5597.9 1956.75  5894.2 1971.94
#Mann= 12 ,-1 , 0
    2671     .07       0  2856.6     .12       0  2945.5     .07       0
  3435.2     .12       0  3565.6     .05       0  3877.9     .07       0
  4079.6     .05       0  4204.6     .07       0  4514.7     .12       0
  4939.1     .04       0  5027.2     .12       0  5189.2     .12       0
Bank Sta=4939.1,5027.2
XS Rating Curve= 0 ,0
Exp/Cntr=0.3,0.1

Type RM Length L Ch R = 1 ,2293902 ,1470,1470,1470
BEGIN DESCRIPTION:
Guadalupe River - 197
END DESCRIPTION:
XS GIS Cut Line= 2
      1851857.43     13935310.83      1853776.38     13932295.33
#Sta/Elev= 30
  2465.9 1923.29    2509 1922.39  2722.8 1916.87  3011.5    1894    3163 1862.36
  3207.7 1846.16  3220.6 1830.94  3232.6 1831.03    3257 1832.52  3302.5 1810.98
  3344.1 1806.29    3450 1801.04  4157.7 1803.41  4345.7 1802.56  4378.2 1803.38
  4439.8 1803.92  4533.8 1788.17  4574.7  1788.5  4815.7 1793.09  4873.3 1780.24
  4895.8 1774.21  4943.3 1777.29  5127.9 1779.42  5154.5 1786.81  5191.6  1806.5
  5222.1 1828.51  5234.6 1851.42  5531.1 1942.43  5770.7 1988.21  6040.2 2014.74
#Mann= 13 ,-1 , 0
  2465.9     .07       0    2509     .12       0  2722.8     .07       0
  3232.6     .12       0  3344.1     .07       0    3450     .05       0
  4157.7     .07       0  4345.7     .05       0  4378.2     .07       0
  4574.7     .05       0  4873.3     .04       0  4943.3     .05       0
  5154.5     .12       0
Bank Sta=4873.3,4943.3
XS Rating Curve= 0 ,0
Exp/Cntr=0.3,0.1

Type RM Length L Ch R = 1 ,2292432 ,1299,1299,1299
XS GIS Cut Line= 3
   1851957.8218613935243.3147222  1853398.79404413934453.3842154
 1854015.113677513934010.6757832
#Sta/Elev= 30
       0 1920.75  328.66 1906.31  517.88  1892.2  687.19 1872.44  756.91 1855.48
  776.83 1841.48  786.79 1839.31   806.7  1840.9  816.66 1837.59  836.58 1824.26
  886.38 1806.62  916.26 1805.32  976.01 1801.11 1075.61 1799.07 1603.45 1796.57
 1713.18 1791.86 1743.13 1777.29 1753.12 1774.71 1872.94 1773.87 1902.89 1778.82
 1942.83 1783.96 2002.74 1783.86 2022.71 1786.31 2042.68 1793.68 2062.65 1805.22
 2152.51 1870.12 2262.34 1938.77 2312.27 1981.33 2342.22  1988.7 2402.13 1991.06
#Mann= 7 ,-1 , 0
       0     .11       0  328.66     .12       0  916.26     .06       0
 1603.45     .12       0 1743.13     .04       0 1902.89     .07       0
 2022.71     .12       0
Bank Sta=1743.13,1902.89
XS Rating Curve= 0 ,0
Exp/Cntr=0.3,0.1

Type RM Length L Ch R = 1 ,2291133 ,1564,1564,1564
BEGIN DESCRIPTION:
Guadalupe River - 196
END DESCRIPTION:
XS GIS Cut Line= 4
      1852644.42     13936281.78      1853516.83     13935582.98
      1854007.28     13935257.46      1854961.06     13934607.15
#Sta/Elev= 30
  3655.2 1921.03  3945.1 1906.59  3994.7 1900.26    4173 1891.19  4343.6 1879.16
  4444.5 1862.92  4457.3 1860.27  4527.7 1823.17  4578.4  1801.8  4626.7 1797.94
  4723.5 1797.04  4906.9 1795.31  4914.8 1792.94    4937 1775.58  4951.5 1772.49
  4966.1 1770.65  4967.6 1769.45  5064.1 1770.65  5066.3 1777.14  5102.3 1779.57
  5282.7 1784.51  5591.4 1779.14  5955.6  1798.8  5980.3 1801.06  6010.1 1813.31
  6060.8 1841.92  6145.6 1898.03  6181.9 1914.63  6369.2 1942.92    6516 1955.11
#Mann= 10 ,-1 , 0
  3655.2     .12       0    4173     .07       0  4444.5     .05       0
  4626.7     .07       0  4723.5     .05       0  4951.5     .07       0
  4966.1     .05       0  5064.1     .12       0  5282.7     .05       0
  5955.6     .12       0
#XS Ineff= 2 , 0
       0                 5515.39       0 1801.35
Permanent Ineff=
       F       F
Bank Sta=4966.1,5064.1
XS Rating Curve= 0 ,0
Exp/Cntr=0.3,0.1

Type RM Length L Ch R = 1 ,2289569 ,2436,2436,2436
BEGIN DESCRIPTION:
Guadalupe River - 195
END DESCRIPTION:
XS GIS Cut Line= 2
      1853523.34     13936976.66      1855526.63     13935837.95
#Sta/Elev= 30
    3478 1907.68  3658.4 1891.55  3736.5 1887.25  3876.4 1869.84  4016.2 1825.84
  4066.6  1819.4  4112.6 1810.17  4140.2 1798.31  4182.1 1796.75  4269.3 1788.87
  4413.2 1790.14  4440.4 1791.41  4823.5 1788.35  4875.3  1780.4  4925.9 1770.26
  4950.7 1765.93  5049.8 1769.42  5071.5 1775.84  5124.8 1778.28  5205.3 1774.18
  5232.9 1782.79    5292 1816.97  5313.7 1824.18  5372.8 1863.02    5416 1885.39
  5496.7 1945.77  5504.4 1971.67  5512.6 1977.07  5571.7 1986.67  5782.3    1999
#Mann= 10 ,-1 , 0
    3478     .12       0  3658.4     .07       0  4066.6     .05       0
  4182.1     .07       0  4269.3     .05       0  4413.2     .07       0
  4440.4     .05       0  4875.3     .07       0  4925.9     .04       0
  5049.8     .12       0
Bank Sta=4925.9,5049.8
XS Rating Curve= 0 ,0
Exp/Cntr=0.3,0.1

Type RM Length L Ch R = 1 ,2287133 ,1875,1875,1875
BEGIN DESCRIPTION:
Guadalupe River - 194
END DESCRIPTION:
XS GIS Cut Line= 2
      1854240.28      13938726.9      1856707.48     13937777.97
#Sta/Elev= 30
  3140.7 1895.01  3186.7 1893.06  3377.7 1887.63  3447.6 1880.97  3524.1 1870.55
  3586.2 1846.93  3595.1 1842.78  3681.5 1800.68    3735 1790.83    3809 1789.17
  3898.3 1789.07  3935.3 1789.18  4378.9 1780.58  4512.3 1782.02    4723 1784.92
  4839.9 1772.98  4878.6 1770.24  4902.9 1765.46  4929.3 1757.38    5010 1760.83
  5086.2 1764.92  5181.4 1799.98  5220.1 1827.41  5225.5 1856.74    5235 1872.59
  5310.1 1911.41  5364.8 1927.99  5474.1 1944.27  5613.3 1955.23  5784.1 1950.87
#Mann= 15 ,-1 , 0
  3140.7     .07       0  3186.7     .12       0  3377.7     .07       0
  3447.6     .12       0  3586.2     .07       0  3595.1     .12       0
    3809     .07       0  3898.3     .12       0  3935.3     .07       0
  4378.9     .05       0  4512.3     .07       0  4839.9     .05       0
  4878.6     .12       0  4902.9     .04       0    5010     .12       0
Bank Sta=4902.9,5010
XS Rating Curve= 0 ,0
Exp/Cntr=0.3,0.1

Type RM Length L Ch R = 1 ,2285258 ,2024,2024,2024
BEGIN DESCRIPTION:
Guadalupe River - 193
END DESCRIPTION:
XS GIS Cut Line= 4
      1854514.44      13940181.9      1855568.76     13940139.72
      1857065.94     13938958.85      1856897.51     13938158.79
#Sta/Elev= 30
  3146.5 1963.56  3244.2 1961.74  3367.2 1955.79  3477.3 1938.23  4069.1 1804.47
  4216.7 1787.72  4485.3 1784.41  4715.6 1781.44  4855.8 1783.76  4878.8 1777.63
  4899.7 1763.46  4911.3 1756.68  4943.7 1755.48  4992.7 1756.68  5021.6 1764.65
  5050.2 1771.45  5167.1 1772.71  5222.9 1771.86  5555.4 1770.94  5805.8 1783.77
  5833.2 1785.65  6004.4 1852.66  6039.7 1853.85  6060.5 1866.16  6132.5 1886.62
  6137.7 1883.21  6232.2 1902.88  6470.1 1927.72  6720.2 1940.47  6926.1 1942.81
#Mann= 12 ,-1 , 0
  3146.5     .07       0  3244.2     .12       0  4069.1     .07       0
  4485.3     .12       0  4715.6     .07       0  4855.8     .12       0
  4899.7     .04       0  5021.6     .12       0  5167.1     .05       0
  5222.9     .06       0  5805.8     .07       0  5833.2     .12       0
Bank Sta=4899.7,5021.6
XS Rating Curve= 0 ,0
Exp/Cntr=0.3,0.1

Type RM Length L Ch R = 1 ,2283234 ,2054,2054,2054
BEGIN DESCRIPTION:
Guadalupe River - 192
END DESCRIPTION:
XS GIS Cut Line= 4
      1857593.13     13941953.24       1857297.9      13941151.9
      1857909.42     13939507.11      1858415.47     13938979.98
#Sta/Elev= 30
    4010 1932.34  4071.8 1926.89  4304.8 1887.82  4486.7 1870.25  4590.2 1857.58
  4696.3 1842.58  4722.1 1832.69  4770.6 1838.45  4819.2 1836.74    4864  1817.6
    4868  1809.2  4923.4 1773.56  4959.1 1759.66  4977.3 1752.37  5025.3 1750.97
  5044.8 1756.69  5218.4 1762.52  5412.7 1775.59  5984.9 1774.37    6009 1774.53
  6187.3 1778.45  6462.7 1780.43  6549.5 1782.92  6566.4 1783.83  6666.6 1790.44
  6779.8 1810.46  7013.1 1886.25  7091.1  1906.8  7197.1 1922.44  7349.5 1929.99
#Mann= 14 ,-1 , 0
    4010     .07       0  4486.7     .05       0  4590.2     .12       0
  4696.3     .05       0  4819.2     .07       0  4959.1     .04       0
  5044.8     .07       0  5218.4     .06       0  5984.9     .07       0
    6009     .06       0  6187.3     .06       0  6462.7     .12       0
  6549.5     .07       0  6566.4     .12       0
Bank Sta=4959.1,5044.8
XS Rating Curve= 0 ,0
Exp/Cntr=0.3,0.1

Type RM Length L Ch R = 1 ,2281180 ,1348,1348,1348
BEGIN DESCRIPTION:
Guadalupe River - 191
END DESCRIPTION:
XS GIS Cut Line= 3
      1858816.16     13942058.65      1859174.64     13941426.03
      1859090.29     13938663.64
#Sta/Elev= 30
  3691.3  1961.1  3824.2 1945.85    3929 1927.68  3995.1 1914.46  4104.1 1893.05
  4463.8 1847.56  4472.7 1846.53  4599.5 1827.46  4696.4 1789.76  4769.6 1759.61
  4789.6 1755.64  4929.7 1752.98  4955.5 1750.11  5019.7 1755.22  5146.8 1762.19
  5279.9 1765.72  5459.9 1759.62  5559.5 1763.93    5600  1772.9  5714.6 1773.17
  5874.7 1773.71  6052.6 1772.98  6151.1 1773.29  6249.6 1780.07  6300.3 1789.82
  6340.4 1806.29  6420.4 1860.02  6470.4 1875.52  7034.3  1916.1  7182.1  1918.7
#Mann= 16 ,-1 , 0
  3691.3     .07       0    3929     .12       0  3995.1     .12       0
  4463.8     .05       0  4472.7     .12       0  4696.4     .07       0
  4929.7     .04       0  5019.7     .07       0  5146.8     .06       0
  5559.5     .07       0  5714.6     .12       0  5874.7     .05       0
  6052.6     .12       0  6151.1     .05       0  6249.6     .12       0
  7034.3     .07       0
Bank Sta=4929.7,5019.7
XS Rating Curve= 0 ,0
Exp/Cntr=0.3,0.1

Type RM Length L Ch R = 1 ,2279832 ,1669,1669,1669
BEGIN DESCRIPTION:
Guadalupe River - 190
END DESCRIPTION:
XS GIS Cut Line= 4
      1860756.18     13941742.38      1859933.77     13939591.46
      1860018.12     13938937.76      1859365.89     13938348.65
#Sta/Elev= 30
  3804.6 1936.71  4153.8 1919.01  4238.7 1908.13  4347.8 1873.44  4498.5 1812.83
  4638.1 1791.21  4687.5 1768.12  4717.5 1759.58  4759.4 1756.58    4942 1757.39
  4966.7  1753.9  4970.1 1748.53    5020 1747.13  5066.8 1748.53  5097.2 1756.41
  5189.2 1768.34  5328.1  1770.5  5756.7 1772.53  5783.7 1772.33  6175.5  1767.9
  6329.8 1770.98  6436.6 1779.02  6471.8 1788.24  6544.6 1830.18  6549.6 1827.56
    6618 1871.28  6768.9 1869.47  6821.3 1869.98  7372.6 1881.41  7645.4 1894.85
#Mann= 13 ,-1 , 0
  3804.6     .12       0  4759.4     .05       0    4942     .04       0
  5097.2     .05       0  5189.2     .05       0  5328.1     .07       0
  5756.7     .05       0  5783.7     .07       0  6175.5     .05       0
  6329.8     .07       0  6471.8     .12       0  6768.9     .07       0
  6821.3     .12       0
Bank Sta=4942,5097.2
XS Rating Curve= 0 ,0
Exp/Cntr=0.3,0.1

Type RM Length L Ch R = 1 ,2278163 ,2196,2196,2196
BEGIN DESCRIPTION:
Guadalupe River - 189
END DESCRIPTION:
XS GIS Cut Line= 3
      1862928.09     13940561.45      1862126.82     13940350.59
      1859533.14     13938452.78
#Sta/Elev= 30
  2939.8 1981.48  3439.3 1955.68  3584.1 1938.14  3646.1 1924.58  3692.4 1907.19
  3902.8 1809.37  4003.1 1786.11  4541.3 1775.23  4839.3  1769.2  4847.8 1760.64
    4854 1762.28  4868.7 1740.68  4892.2 1738.84  5010.7  1740.8  5046.9 1754.02
    5076 1754.26  5232.8 1757.03  5326.5 1766.83  5472.1 1766.26  5790.6  1766.3
  5979.3 1777.52  6035.3 1785.25  6106.3 1811.34  6156.5 1840.14  6188.2 1845.29
  6327.9 1847.63  6426.9 1861.45  6442.9 1868.18  6620.6 1880.61  6982.2  1890.5
#Mann= 9 ,-1 , 0
  2939.8     .12       0  4541.3     .07       0  4868.7     .04       0
  5010.7     .07       0    5076     .07       0  5472.1     .05       0
  5979.3     .12       0  6188.2     .07       0  6426.9     .12       0
Bank Sta=4868.7,5010.7
XS Rating Curve= 0 ,0
Exp/Cntr=0.3,0.1

Type RM Length L Ch R = 1 ,2275967 ,2002,2002,2002
BEGIN DESCRIPTION:
Guadalupe River - 188
END DESCRIPTION:
XS GIS Cut Line= 3
      1863370.98     13939317.36      1861726.17     13937609.28
      1860671.79     13937314.06
#Sta/Elev= 30
  2850.8 1960.59  2927.3 1963.32  2960.5 1961.76  2998.1 1958.54  3068.9 1941.67
  3231.4 1888.41  3429.5 1797.58    3456    1796  3486.1 1779.02  3585.2 1768.25
  3805.9 1764.21  3862.4 1763.64  4092.9 1764.63    4648 1759.16  4832.7 1753.22
  4872.3 1752.24  4907.8 1739.41    4943  1741.4  5007.9 1735.24  5091.5 1740.37
  5127.7 1748.94  5204.7 1793.01  5314.1 1800.68  5653.7 1826.98  5732.1  1837.2
  5790.5 1851.42  5847.9 1861.08  5908.7 1877.02  6065.6 1893.91    6317 1906.13
#Mann= 17 ,-1 , 0
  2850.8     .08       0  2927.3     .05       0  2960.5     .12       0
    3456     .05       0  3805.9     .07       0  3862.4     .05       0
  4092.9     .07       0    4648     .12       0  4832.7     .07       0
    4943     .04       0  5091.5     .07       0  5127.7     .12       0
  5314.1     .05       0  5653.7     .07       0  5790.5     .12       0
  5847.9     .07       0  6065.6     .05       0
Bank Sta=4943,5091.5
XS Rating Curve= 0 ,0
Exp/Cntr=0.3,0.1

Type RM Length L Ch R = 1 ,2273965 ,3681,3681,3681
BEGIN DESCRIPTION:
Guadalupe River - 187
END DESCRIPTION:
XS GIS Cut Line= 6
      1863516.03     13939702.96      1863601.48     13937575.01
      1863628.13     13937231.33      1864100.23     13936124.17
      1863916.44     13935603.44      1863501.62      13934243.6
#Sta/Elev= 30
  2722.2 1946.54  2786.3 1937.54  2880.3 1918.03  2940.3 1915.03  3180.5 1933.97
  3270.6 1932.49  3474.4 1894.17  3769.3 1832.54  3867.6 1816.84  3901.1  1806.2
  3965.9 1804.54  4002.4 1804.35  4051.2 1799.99  4121.3 1774.66  4171.3 1769.03
  4841.9 1754.51  4931.2  1742.9  4952.2 1737.78  5026.2 1729.47  5042.4 1736.93
  5569.7 1743.26  5845.7 1758.87  6302.4 1760.22  6829.9 1775.08  6917.6 1778.39
  7143.3 1799.73  7248.7 1813.71  7385.2 1850.23  7827.5 1916.76  8374.1  1922.5
#Mann= 16 ,-1 , 0
  2722.2     .07       0  2786.3     .12       0  3474.4     .05       0
  3769.3     .12       0  3867.6     .05       0  3965.9     .07       0
  4002.4     .05       0  4931.2     .07       0  4952.2     .04       0
  5042.4     .07       0  5569.7     .05       0  5845.7     .07       0
  6302.4     .05       0  6829.9     .12       0  6917.6     .07       0
  7143.3     .12       0
Bank Sta=4952.2,5042.4
XS Rating Curve= 0 ,0
Exp/Cntr=0.3,0.1

Type RM Length L Ch R = 1 ,2270284 ,1552,1552,1552
BEGIN DESCRIPTION:
Guadalupe River - 186
END DESCRIPTION:
XS GIS Cut Line= 6
      1867506.06     13937931.12      1867063.27     13936764.93
      1865735.33     13936174.73      1864847.35     13935449.75
      1864801.32     13935425.92      1863949.06      13934187.3
#Sta/Elev= 30
  3011.2 1856.99  3305.6 1847.41  3449.3 1830.68  3685.6 1812.63  4005.1 1794.81
  4046.3 1793.64  4100.3 1792.11    4156 1790.54    4202 1780.43  4323.9 1759.05
  4735.7 1747.09  4834.2 1731.03  4927.6 1731.48  4983.9 1721.85  5077.5 1730.49
  5106.4 1739.82  5181.6 1744.06  5233.6 1736.43  5477.1 1737.94  5742.1 1755.33
  6176.2 1757.52  6848.3 1764.44  7031.1 1776.35  7404.5 1824.91  7680.3 1902.26
    7936 1959.52  8043.7 1973.27  8159.8 1975.12  8365.4 1975.46  8413.5 1974.66
#Mann= 15 ,-1 , 0
  3011.2     .05       0  3449.3     .08       0  3685.6     .05       0
  4005.1     .07       0  4046.3     .05       0  4100.3     .12       0
    4202     .05       0  4927.6     .04       0  5077.5     .05       0
  5742.1     .06       0  6176.2     .05       0  7680.3     .12       0
    7936     .08       0  8159.8     .12       0  8365.4     .05       0
Bank Sta=4927.6,5077.5
XS Rating Curve= 0 ,0
Exp/Cntr=0.3,0.1

Type RM Length L Ch R = 1 ,2268732 ,2173,2173,2173
BEGIN DESCRIPTION:
Guadalupe River - 185
END DESCRIPTION:
XS GIS Cut Line= 4
      1868133.79     13938205.17      1867417.63     13935318.84
      1866375.97     13934103.57      1866419.37     13933474.22
#Sta/Elev= 30
  2341.4 1890.61  2409.5 1878.78  2579.7 1837.06  2741.2 1815.04  2816.5 1809.43
  3520.6 1793.62  3843.6 1775.69  3969.5  1768.5  4058.4 1752.35  4316.3 1750.31
  4477.7  1747.1  4579.9  1745.1  4824.6 1737.74  4973.2 1730.61  5075.5 1720.96
  5133.7 1726.49    5227 1731.35  5404.9 1724.61  5454.2 1731.96  5511.3  1753.9
  6071.1 1765.06  6141.3 1773.29  6242.3 1802.95  6549.3 1942.25  6589.1 1959.26
  6652.8 1964.91  6840.4 1964.59  6866.9 1964.81  7164.3 1951.04  7546.7 1970.01
#Mann= 17 ,-1 , 0
  2341.4     .07       0  2409.5     .12       0  2579.7     .05       0
  2741.2     .12       0  2816.5     .07       0  3843.6     .05       0
  4316.3     .07       0  4477.7     .12       0  4579.9     .05       0
  4824.6     .12       0  4973.2     .04       0  5133.7     .12       0
  6141.3     .12       0  6549.3     .05       0  6840.4     .12       0
  6866.9     .05       0  7164.3     .12       0
Bank Sta=4973.2,5133.7
XS Rating Curve= 0 ,0
Exp/Cntr=0.3,0.1

Type RM Length L Ch R = 1 ,2266559 ,2037,2037,2037
BEGIN DESCRIPTION:
Guadalupe River - 184
END DESCRIPTION:
XS GIS Cut Line= 6
      1868802.48     13937758.33      1868824.83     13936552.13
      1868909.39     13935621.86      1868961.66     13935047.11
      1868893.94     13934767.24      1868716.22     13933308.71
#Sta/Elev= 30
  2574.4 1815.08  2857.8 1796.74  3112.4 1790.53  3317.9  1788.6  3567.9 1775.98
  3717.9 1750.09  3824.8 1743.66    4039 1749.65  4556.8 1747.33  4655.3  1745.8
  4714.9 1743.51  4753.8 1731.22  4842.3 1725.51    4973 1720.86  5123.5 1725.96
  5183.7 1738.87  5269.6 1788.06  5346.5  1804.2    5388 1811.39    5493 1845.49
  5622.5 1877.74  5778.3 1894.53  5884.5 1883.56  6024.3 1847.23  6104.8 1829.06
  6247.4 1835.99  6691.4 1881.92  6791.1 1879.32  6980.6 1843.15  7049.3 1827.16
#Mann= 12 ,-1 , 0
  2574.4     .12       0  3112.4     .05       0  4556.8     .07       0
  4655.3     .05       0  4753.8     .12       0  4842.3    .035       0
  5123.5     .05       0  5346.5     .12       0    5493     .07       0
  6024.3     .12       0  6247.4     .07       0  6980.6     .05       0
Bank Sta=4842.3,5123.5
XS Rating Curve= 0 ,0
Exp/Cntr=0.3,0.1

Type RM Length L Ch R = 1 ,2264522 ,1557,1557,1557
BEGIN DESCRIPTION:
Guadalupe River - 183
END DESCRIPTION:
XS GIS Cut Line= 3
      1870043.51     13937966.39      1870824.75     13934016.76
      1871106.66     13933409.57
#Sta/Elev= 30
  2612.4 1832.09  3062.8 1798.22  3211.5 1793.02  3472.8 1796.79    3595 1788.83
  3827.9 1770.24    3830 1770.22  3993.5 1760.78  4344.1 1738.41    4622 1739.63
  4773.1 1722.09  4846.3 1729.13  4948.2 1724.04  4988.2 1717.97  5090.9 1724.01
  5126.3 1726.44  5161.3 1727.35  5366.1 1719.97  5425.5 1745.91  5525.4 1755.73
  5551.7 1758.37  5738.1 1770.59  5936.3 1794.11  6085.6 1823.56  6395.7 1909.54
    6512  1928.9  6791.4 1934.61  6980.1 1942.74  7059.8    1953    7308 1960.91
#Mann= 14 ,-1 , 0
  2612.4     .12       0    3595     .07       0  3827.9     .05       0
    3830     .07       0  3993.5     .05       0  4773.1     .07       0
  4948.2     .04       0  5090.9     .12       0  5126.3     .05       0
  5161.3     .07       0  5525.4     .12       0  5551.7     .05       0
  5936.3     .07       0  6085.6     .12       0
Bank Sta=4948.2,5090.9
XS Rating Curve= 0 ,0
Exp/Cntr=0.3,0.1

Type RM Length L Ch R = 1 ,2262965 ,2496,2496,2496
BEGIN DESCRIPTION:
Guadalupe River - 182
END DESCRIPTION:
XS GIS Cut Line= 6
      1870754.27     13937887.99       1871619.2     13936601.28
      1872334.47     13935061.68      1872340.36     13935007.28
      1872363.93     13934788.52      1872540.15      13933511.1
#Sta/Elev= 30
  3144.7 1815.11  3149.2 1815.11  3241.4 1810.86  3357.4 1805.87  3705.3 1792.68
  3706.1 1792.65  3940.6 1779.12  4077.4 1781.12  4401.4 1768.54  4436.9 1765.91
  4801.3 1739.76  4839.3 1724.68  4934.7 1716.07  4982.5 1712.71  5017.7 1706.24
  5065.9 1712.56  5279.4 1717.92  5493.1 1719.17  5647.2 1735.28  6194.2 1751.43
  6423.1 1781.22  6628.3 1815.86    6858 1890.05  7034.4 1933.61  7366.5 1948.08
    7744 1930.89  7808.1 1921.23  7893.9 1891.61  7912.7 1885.76    7957 1894.21
#Mann= 19 ,-1 , 0
  3144.7     .07       0  3149.2     .05       0  3241.4     .12       0
  3357.4     .05       0  3705.3     .07       0  3706.1     .05       0
  4077.4     .12       0  4401.4     .08       0  4436.9     .05       0
  4839.3     .12       0  4934.7     .05       0  4982.5     .04       0
  5065.9     .05       0  5279.4     .07       0  5493.1     .12       0
  5647.2     .05       0  6423.1     .12       0    7744     .07       0
  7893.9     .12       0
Bank Sta=4982.5,5065.9
XS Rating Curve= 0 ,0
Exp/Cntr=0.3,0.1

Type RM Length L Ch R = 1 ,2260469 ,1898,1898,1898
BEGIN DESCRIPTION:
Guadalupe River - 181
END DESCRIPTION:
XS GIS Cut Line= 3
      1873277.01     13938552.35      1874318.68     13934884.82
      1873950.21     13933779.41
#Sta/Elev= 30
  3076.4 1913.59  3161.3 1911.33  3245.1 1900.51  3380.2  1880.6  3395.9 1869.25
  3453.2 1851.79  3559.2 1833.95  3750.3 1811.78    3937 1793.84  4156.3 1782.09
  4268.4 1773.92  4373.3 1774.62  4441.1 1747.62  4572.4 1735.76  4673.7 1732.59
  4845.1 1722.99  4892.9 1711.09  4958.1 1704.79  5048.8 1711.39  5760.1 1747.39
  6012.9 1783.98  6194.9 1798.58  6424.3 1814.31  6708.9 1886.23  6886.3 1909.24
  7105.5 1908.64  7332.2  1884.6  7553.5 1895.59  7689.9 1910.78  8054.2 1925.87
#Mann= 13 ,-1 , 0
  3076.4     .07       0  3245.1     .05       0  3559.2     .07       0
  3750.3     .05       0    3937     .12       0  4156.3     .05       0
  4268.4     .12       0  4572.4     .07       0  4673.7     .05       0
  4892.9     .04       0  5048.8     .05       0  6194.9     .05       0
  6424.3     .12       0
Bank Sta=4892.9,5048.8
XS Rating Curve= 0 ,0
Exp/Cntr=0.3,0.1

Type RM Length L Ch R = 1 ,2258571 ,593,593,593
BEGIN DESCRIPTION:
Guadalupe River - 180
END DESCRIPTION:
XS GIS Cut Line= 6
       1875262.9     13938449.71      1875409.41     13936682.88
       1875479.4     13936490.46      1875116.14     13935729.32
      1875128.69     13935659.05      1874557.07      13933883.5
#Sta/Elev= 30
  2746.3 1839.23  3173.5 1793.06  3416.1 1777.87  3607.7 1765.76  3737.8 1760.64
  4337.7 1738.17  4583.1 1729.73  4623.3 1739.69  4746.2  1737.8  4785.4 1722.88
  4865.2 1722.21    4905 1708.17  5042.7 1705.79  5086.4 1710.09  5175.7 1714.27
  5507.7 1732.98  5613.2 1738.31  5820.7  1797.1  5925.1 1802.36  6063.3 1806.65
  6389.5  1877.1  6490.3 1889.07  6549.9 1888.33  6655.9 1864.35  6710.3 1839.59
  6819.6 1881.24  6969.1 1904.54  7169.8 1911.66  7378.5 1887.04    7504 1850.72
#Mann= 19 ,-1 , 0
  2746.3     .12       0  3173.5     .07       0  3416.1     .12       0
  3607.7     .07       0  3737.8     .05       0  4337.7     .07       0
  4583.1     .05       0    4905    .035       0  5086.4    .035       0
  5175.7     .05       0  5507.7     .07       0  5613.2     .12       0
  5820.7     .05       0  5925.1     .08       0  6063.3     .12       0
  6490.3     .08       0  6655.9     .07       0  6969.1     .05       0
  7378.5     .12       0
Bank Sta=4905,5086.4
XS Rating Curve= 0 ,0
Exp/Cntr=0.3,0.1

Type RM Length L Ch R = 1 ,2257978 ,1609,1609,1609
XS GIS Cut Line= 4
  1876260.80934313937437.3162396  1876405.14173213936063.0214161
 1875564.249056813935874.7619501 1874924.166675613934864.4355586
#Sta/Elev= 30
       0 1772.94  298.24 1765.87  497.07 1750.37  656.13 1744.41 1202.91 1732.84
 1302.32  1727.2 1352.03 1722.16 1411.57 1721.34 1451.19 1712.11 1560.14 1709.57
 1621.09 1700.92 1664.06 1700.92  1688.9 1706.29 1738.42 1707.66 1966.23 1706.69
 2243.56 1720.98 2313.33  1727.8 2492.73 1731.72  2592.4 1737.74 2751.87 1778.91
 2781.77 1783.15 2891.41 1786.63 2921.31 1785.06 2961.18 1778.92 3020.98 1780.33
 3050.88 1787.43 3110.68 1794.07 3170.48 1804.74 3280.12 1838.24 3439.59  1871.7
#Mann= 7 ,-1 , 0
       0     .12       0  656.13     .08       0 1302.32     .05       0
 1411.57      .1       0 1560.14     .04       0 1738.42      .1       0
 2243.56     .12       0
Bank Sta=1560.14,1738.42
XS Rating Curve= 0 ,0
Exp/Cntr=0.3,0.1

Type RM Length L Ch R = 1 ,2256369 ,2374,2374,2374
BEGIN DESCRIPTION:
Guadalupe River - 179
END DESCRIPTION:
XS GIS Cut Line= 3
      1875946.29     13938422.12      1877356.87     13934754.61
      1878267.26     13934169.36
#Sta/Elev= 30
  1883.5 1829.14  1929.2  1823.2  2061.3 1811.64  2246.5  1800.9  2253.8 1800.33
  2349.8 1796.67  2501.6 1790.94  2829.2 1773.56    3258 1754.88  3400.2 1756.82
  3738.4 1740.37  4084.4 1733.42  4232.9 1731.02  4545.2 1713.85  4649.2 1713.47
  4857.4 1707.92  4998.2 1699.24  5031.2 1693.53  5105.4 1699.98  5262.6 1700.64
  5341.1 1723.97  5397.8 1753.12  5501.8 1808.38  5571.2 1867.86  5587.5 1896.43
  5608.9 1912.36  5685.8 1936.88  5876.5 1947.76  6557.4 1935.14  6895.2 1955.71
#Mann= 18 ,-1 , 0
  1883.5     .12       0  1929.2     .05       0  2061.3     .12       0
  2246.5     .05       0  2253.8     .12       0  2349.8     .05       0
  2501.6     .07       0  2829.2     .12       0  3400.2     .05       0
  3738.4     .12       0  4084.4     .07       0  4232.9     .05       0
  4545.2     .12       0  4649.2     .05       0  4857.4     .08       0
  4998.2     .04       0  5105.4     .08       0  5397.8     .12       0
Bank Sta=4998.2,5105.4
XS Rating Curve= 0 ,0
Exp/Cntr=0.3,0.1

Type RM Length L Ch R = 1 ,2253995 ,3258,3258,3258
BEGIN DESCRIPTION:
Guadalupe River - 178
END DESCRIPTION:
XS GIS Cut Line= 6
      1878007.92     13938769.32      1878399.53     13937112.03
      1878851.87     13936249.67      1878972.78     13936019.22
      1879112.47     13935752.89      1879244.86     13934559.62
#Sta/Elev= 30
  2212.9 1807.07  2303.8 1802.54  2834.7 1785.22  2857.7 1784.92  3058.3 1778.92
  3158.6 1776.44  3258.9 1773.46  3660.1 1759.44  3727.8 1738.61  3785.9 1732.39
  4012.5 1726.47  4183.5 1725.62  4351.6 1721.92  4503.8  1720.6  4793.3 1704.17
  4825.4 1696.28  4954.1 1693.74  4994.6  1697.4  5057.2 1718.23  5140.8 1729.23
    5439 1743.52    5539 1756.59  5609.6  1777.2  5788.2 1844.33  5969.5 1904.08
  5974.5 1901.88  6150.7 1965.35  6223.2  1978.2  6315.5 1983.51  6651.2 1981.26
#Mann= 18 ,-1 , 0
  2212.9     .05       0  2303.8     .07       0  2834.7     .05       0
  2857.7     .07       0  3058.3     .12       0  3158.6     .07       0
  3258.9     .12       0  3660.1     .05       0  4012.5     .08       0
  4183.5     .12       0  4351.6     .05       0  4503.8     .12       0
  4825.4     .04       0  4994.6     .12       0  5057.2     .05       0
    5439     .07       0  5609.6     .12       0  6315.5     .07       0
Bank Sta=4825.4,4994.6
XS Rating Curve= 0 ,0
Exp/Cntr=0.3,0.1
