--- Rough Hollow.prj (project) ---

Proj Title=Rough Hollow Base Level Engineering
Current Plan=p01
Default Exp/Contr=0.3,0.1
English Units
Geom File=g01
Flow File=f01
Plan File=p01
Y Axis Title=Elevation
X Axis Title(PF)=Main Channel Distance
X Axis Title(XS)=Station
BEGIN DESCRIPTION:
Rough Hollow
END DESCRIPTION:
DSS Export Rating Curves= 0
DSS Export Rating Curve Sorted= 0
DSS Export Volume Flow Curves= 0
DXF OffsetX= 0
DXF OffsetY= 0
DXF ScaleX= 1
DXF ScaleY= 10

--- Rough Hollow.p01 (plan) ---

Plan Title=Multiple Run
Short Identifier=Multiple
Geom File=g01
Flow File=f01
Subcritical Flow
K Sum by GR= 0
Std Step Tol= 0.01
Critical Tol= 0.01
Num of Std Step Trials= 20
Max Error Tol= 0.3
Flow Tol Ratio= 0.001
Split Flow NTrial= 30
Split Flow Tol= 0.02
Split Flow Ratio= 0.02
Log Output Level= 0
Friction Slope Method= 1
Unsteady Friction Slope Method= 2
Unsteady Bridges Friction Slope Method= 1
Parabolic Critical Depth
Global Vel Dist=  1 , 1 , 1
Global Log Level= 0
CheckData=True
Encroach Param= -1, 0, 0, 0
BEGIN DESCRIPTION:
Multiple Run
END DESCRIPTION:

--- Rough Hollow.f01 (steady flow) ---

Flow Title=Multiple
Number of Profiles=7
Profile Names=10-year,25-year,50-year,1pct_min,100-year,1pct_plu,500-year
River Rch & RM= Rough Hollow,Reach-1,28789
    2099    3695    5256    3601    7185   14337   13290
River Rch & RM= Rough Hollow,Reach-1,22620
    4754    8625   12513    8720   17398   34714   33298
River Rch & RM= Rough Hollow,Reach-1,15546
    5778   10550   15375   10755   21459   42817   41385
River Rch & RM= Rough Hollow,Reach-1,12315
    5999   10972   16008   11210   22366   44626   43225
River Rch & RM= Rough Hollow,Reach-1,7331
    6095   11148   16264   11388   22723   45338   43909
River Rch & RM= Rough Hollow,Reach-1,6224
    6283   11501   16789   11761   23467   46823   45388
River Rch & RM= Rough Hollow,Reach-1,4672
    6488   11898   17389   12196   24335   48554   47177
Boundary for River Rch & Prof#=Rough Hollow,Reach-1,1
Up Type=0
Dn Type=3
Dn Slope=0.005
Boundary for River Rch & Prof#=Rough Hollow,Reach-1,2
Up Type=0
Dn Type=3
Dn Slope=0.005
Boundary for River Rch & Prof#=Rough Hollow,Reach-1,3
Up Type=0
Dn Type=3
Dn Slope=0.005
Boundary for River Rch & Prof#=Rough Hollow,Reach-1,4
Up Type=0
Dn Type=3
Dn Slope=0.005
Boundary for River Rch & Prof#=Rough Hollow,Reach-1,5
Up Type=0
Dn Type=3
Dn Slope=0.005
Boundary for River Rch & Prof#=Rough Hollow,Reach-1,6
Up Type=0
Dn Type=3
Dn Slope=0.005
Boundary for River Rch & Prof#=Rough Hollow,Reach-1,7
Up Type=0
Dn Type=3
Dn Slope=0.005

--- Rough Hollow.g01 (geometry) ---

Geom Title=Existing Conditions
Program Version=4.10

River Reach=Rough Hollow    ,Reach-1
Reach XY= 30
        1846625.       13996425.      1847115.18     13995885.47
      1847752.48     13995548.33      1848330.26     13994630.47
       1849284.8     13994114.52      1849701.27      13993447.3
        1850375.       13993025.      1850132.32      13992625.1
      1850278.83     13992176.58      1850969.56     13991619.81
      1851124.97     13991259.58      1850616.65     13990578.19
      1850027.05     13990519.16        1849925.       13990075.
      1850271.46     13989723.54      1850324.93     13989195.03
      1849824.51      13987090.2      1849983.14     13986268.94
      1851021.46     13985223.54      1851021.39      13984576.5
      1850588.21     13983988.63      1849488.61     13983288.24
      1848834.98     13981935.69      1847021.77     13981516.75
       1846526.2      13981114.5      1846694.58     13980358.93
      1848376.26     13979099.58      1849204.18     13977954.44
      1849222.21     13977387.49      1848557.74     13976642.26

Type RM Length L Ch R = 1 ,28789   ,410,410,410
BEGIN DESCRIPTION:
Rough Hallow 55.0
END DESCRIPTION:
XS GIS Cut Line= 3
      1847025.01     13996425.01        1846725.       13996225.
      1846575.04     13996125.03
#Sta/Elev= 30
  4639.2 2119.77  4667.8 2119.27  4682.8 2115.97  4688.8 2115.48  4718.8  2110.3
  4739.9 2108.52  4754.9 2108.49    4806 2106.34  4927.7 2104.81  4992.3 2103.44
  5002.8 2102.98  5007.3 2101.15  5019.8 2098.55  5020.2 2098.05  5024.5 2098.05
  5024.9 2098.55  5028.3 2101.46  5035.8 2103.95  5043.3 2104.16  5058.4 2103.03
  5064.4 2103.24  5085.4 2102.34  5115.4 2110.47  5121.5 2111.24  5136.5 2114.33
  5151.5 2118.61  5157.5 2119.03  5165.6 2121.04  5170.3 2121.63    5180 2122.47
#Mann= 5 ,-1 , 0
  4639.2     .07       0  5019.8     .05       0  5024.9     .07       0
  5165.6      .1       0  5170.3     .07       0
Bank Sta=5019.8,5024.9
XS Rating Curve= 0 ,0
Exp/Cntr=0.3,0.1

Type RM Length L Ch R = 1 ,28379   ,457,457,457
BEGIN DESCRIPTION:
Rough Hallow 54.0
END DESCRIPTION:
XS GIS Cut Line= 3
      1847174.98     13996274.97        1847025.       13995975.
      1846624.99       13995875.
#Sta/Elev= 30
  4671.1 2119.45  4707.4 2118.23  4752.1 2113.11  4813.6 2109.08  4858.3 2103.81
    4917 2099.03  4970.1  2100.7  4975.7 2099.06  4981.6 2095.02    4982 2094.52
  4986.7 2095.02  4992.5 2097.11  5003.7 2099.46  5029.7 2099.05    5058 2100.14
  5070.9 2099.38  5099.2 2101.27  5140.5 2102.02  5161.1 2099.88  5171.4 2101.01
  5189.4 2100.93  5212.6 2102.45  5253.9 2102.64  5295.1 2104.01  5318.3 2106.88
  5354.4  2114.8  5387.9 2119.81  5395.6 2121.65  5400.7 2121.45  5418.8 2123.51
#Mann= 3 ,-1 , 0
  4671.1     .07       0  4981.6     .05       0  4986.7     .07       0
Bank Sta=4981.6,4986.7
XS Rating Curve= 0 ,0
Exp/Cntr=0.3,0.1

Type RM Length L Ch R = 1 ,27922   ,601,601,601
BEGIN DESCRIPTION:
Rough Hallow 53.0
END DESCRIPTION:
XS GIS Cut Line= 3
      1847525.01     13996025.02        1847425.       13995825.
      1846925.01     13995075.01
#Sta/Elev= 30
  4772.1 2120.12  4802.9 2117.97  4869.9 2103.36  4897.9 2100.96    4937 2099.16
  4981.8 2094.68  4987.3 2095.81  5003.2 2094.97  5039.3 2096.66  5054.3 2096.24
  5162.5 2097.51  5255.6 2095.78  5289.1 2093.93  5289.5 2093.43  5294.3 2093.93
  5297.7 2095.77  5306.7 2097.31  5428.4  2097.4    5478 2099.03  5508.5 2101.49
  5536.6 2105.45  5565.1  2108.5  5601.2 2111.32  5637.2 2117.23  5652.2 2120.65
  5694.3  2123.4  5738.5 2125.01    5825 2129.61  5868.6  2133.3  5897.1 2134.69
#Mann= 5 ,-1 , 0
  4772.1     .07       0  5289.1     .05       0  5294.3     .07       0
  5508.5      .1       0  5738.5     .07       0
Bank Sta=5289.1,5294.3
XS Rating Curve= 0 ,0
Exp/Cntr=0.3,0.1

Type RM Length L Ch R = 1 ,27321   ,294,294,294
BEGIN DESCRIPTION:
Rough Hallow 52.0
END DESCRIPTION:
XS GIS Cut Line= 3
        1847875.     13995825.03      1847824.72     13995443.62
      1847025.02     13994975.01
#Sta/Elev= 30
  4555.7 2124.16    4586 2121.54  4616.3 2112.54  4686.9 2098.05  4767.6 2093.94
  4896.8 2092.75  4901.9 2090.07  4943.1 2093.41  4946.7 2091.25  4952.5  2092.9
  4962.4 2089.63  4968.2 2092.27  4974.9 2089.69  5005.4 2089.56    5024  2086.9
  5024.5  2086.4  5029.7  2086.9  5032.8  2090.1    5056 2091.98  5202.8 2091.16
    5240 2093.14  5400.2 2094.99  5437.4  2098.5  5458.8  2102.3  5464.6 2104.94
  5480.3 2106.21  5486.1 2108.72  5503.7 2111.23  5658.7  2124.8  5867.3 2135.41
#Mann= 5 ,-1 , 0
  4555.7     .07       0    5024     .05       0  5029.7     .07       0
  5503.7      .1       0  5658.7     .07       0
Bank Sta=5024,5029.7
XS Rating Curve= 0 ,0
Exp/Cntr=0.3,0.1

Type RM Length L Ch R = 1 ,27027   ,442,442,442
BEGIN DESCRIPTION:
Rough Hallow 51.0
END DESCRIPTION:
XS GIS Cut Line= 3
      1848275.02     13995575.03        1847925.       13995175.
      1847525.04     13994875.03
#Sta/Elev= 30
  4468.2 2113.96  4503.8 2110.39  4518.1 2106.81  4546.5 2102.18  4560.8 2101.12
  4610.1 2095.11  4652.8 2092.29  4759.1 2089.28    4837 2089.64  4893.4 2088.29
  4907.2 2089.36  4914.8 2088.46  4943.3 2089.86  4978.4 2089.64  5002.9 2088.62
  5004.2 2087.35  5004.6 2086.85  5009.9 2087.35  5027.9 2089.57    5107 2090.28
  5121.6 2091.22  5171.6 2090.98    5207 2092.11  5236.2 2093.49  5277.9 2097.31
  5321.6  2098.6  5329.2 2099.51  5442.5 2106.59    5490 2108.68  5499.7  2109.5
#Mann= 5 ,-1 , 0
  4468.2     .07       0  5004.2     .05       0  5009.9     .07       0
  5329.2      .1       0    5490     .07       0
Bank Sta=5004.2,5009.9
XS Rating Curve= 0 ,0
Exp/Cntr=0.3,0.1

Type RM Length L Ch R = 1 ,26585   ,448,448,448
BEGIN DESCRIPTION:
Rough Hallow 50.0
END DESCRIPTION:
XS GIS Cut Line= 3
      1848575.01     13995325.02        1848275.       13994925.
      1847875.03     13994725.02
#Sta/Elev= 30
  4495.7 2116.15  4538.4 2114.92    4553 2108.77  4559.3 2108.09  4567.6 2105.87
  4609.3  2098.6  4638.4 2095.94  4659.3 2094.55  4738.4 2092.28  4882.2 2088.72
  4888.4 2089.17  4917.6 2086.11  4959.3 2085.76  4982.2 2083.59  4988.4 2081.19
  4992.6  2078.4  4998.5  2078.4  5004.1 2076.27  5006.8 2076.18  5007.2 2075.68
  5012.6 2076.18  5026.5    2081  5071.2 2083.42  5085.2 2083.25  5107.5 2085.58
  5129.9 2086.66  5308.8 2090.42  5331.1  2091.4  5389.8 2096.13  5442.9 2098.31
#Mann= 3 ,-1 , 0
  4495.7     .07       0  5006.8     .05       0  5012.6     .07       0
Bank Sta=5006.8,5012.6
XS Rating Curve= 0 ,0
Exp/Cntr=0.3,0.1

Type RM Length L Ch R = 1 ,26137   ,872,872,872
BEGIN DESCRIPTION:
Rough Hallow 49.0
END DESCRIPTION:
XS GIS Cut Line= 3
      1848675.02     13994825.02        1848425.       13994575.
      1848067.18     13994289.74
#Sta/Elev= 30
  4646.6 2092.56  4674.9    2092  4703.2 2086.37  4717.3  2084.4  4731.5 2083.26
  4745.6 2083.16  4759.8 2082.33  4816.3 2082.32  4901.2 2080.99  4929.5 2080.92
  4943.6 2081.71  4957.8 2080.51  5003.4 2078.95  5018.9 2073.83  5019.4 2073.33
  5024.3 2073.33  5024.8 2073.83  5028.2 2074.09  5036.2 2087.19  5050.6 2089.52
  5077.8 2090.62  5149.9 2091.39  5199.6 2092.73  5220.4 2092.46  5284.4 2093.15
  5292.4 2093.96  5377.3 2095.53  5398.1 2095.29    5435 2095.85  5457.8 2096.57
#Mann= 3 ,-1 , 0
  4646.6     .07       0  5018.9     .05       0  5024.8     .07       0
Bank Sta=5018.9,5024.8
XS Rating Curve= 0 ,0
Exp/Cntr=0.3,0.1

Type RM Length L Ch R = 1 ,25265   ,480,480,480
BEGIN DESCRIPTION:
Rough Hallow 48.0
END DESCRIPTION:
XS GIS Cut Line= 3
        1849175.     13994425.01        1849125.       13994175.
      1848774.98     13993774.98
#Sta/Elev= 30
  4730.9 2086.54  4751.3 2086.37  4771.7 2083.62  4781.9 2081.22  4792.1 2079.76
  4802.3 2079.24  4812.5 2077.37  4843.1  2076.3  4924.7 2075.15  4955.3 2073.89
  4975.7 2070.21  4983.3 2072.35    4993 2072.96  5021.5 2073.03  5028.1 2072.75
  5039.2 2069.76  5039.7 2069.26  5044.9 2069.26  5045.4 2069.76  5064.2 2073.39
  5078.4 2074.72  5156.2 2076.91  5162.9 2077.61  5262.5 2079.14  5321.7 2081.26
  5354.6 2083.36  5361.2  2084.4  5400.4 2085.91  5489.4 2090.35  5517.4 2090.76
#Mann= 5 ,-1 , 0
  4730.9     .07       0  5039.2     .05       0  5045.4     .07       0
  5321.7      .1       0  5400.4     .07       0
Bank Sta=5039.2,5045.4
XS Rating Curve= 0 ,0
Exp/Cntr=0.3,0.1

Type RM Length L Ch R = 1 ,24785   ,443,443,443
BEGIN DESCRIPTION:
Rough Hallow 47.0
END DESCRIPTION:
XS GIS Cut Line= 3
        1849675.       13994025.        1849425.       13993875.
        1849125.       13993675.
#Sta/Elev= 30
  4703.8 2084.11  4717.4 2083.97  4754.3 2082.47  4820.4 2079.24    4834 2078.21
  4913.7 2074.88    4937 2072.35  4944.8 2069.46  4950.6 2068.16    4972 2069.17
  4981.7 2069.17  4987.6 2068.74  4992.4 2067.71  5014.3 2067.41  5014.8 2066.91
    5021 2066.91  5021.5 2067.41  5031.4 2069.94  5038.9 2070.47  5059.9 2070.77
    5081 2071.89  5168.1 2072.32  5204.2 2072.89  5211.7 2073.27  5240.2 2078.06
  5247.7 2079.09  5255.2 2079.26  5261.3 2080.39  5283.8 2081.45  5355.9 2083.27
#Mann= 3 ,-1 , 0
  4703.8     .07       0  5014.3     .05       0  5021.5     .07       0
Bank Sta=5014.3,5021.5
XS Rating Curve= 0 ,0
Exp/Cntr=0.3,0.1

Type RM Length L Ch R = 1 ,24342   ,412,412,412
BEGIN DESCRIPTION:
Rough Hallow 46.0
END DESCRIPTION:
XS GIS Cut Line= 3
      1849825.01     13993775.01        1849675.       13993525.
      1849274.96     13993374.99
#Sta/Elev= 30
  4704.1 2082.61  4748.8 2080.12  4762.4 2078.65  4785.7 2075.68  4820.7 2069.62
  4834.3 2068.21  4855.7 2067.68  4892.6 2068.86  4923.7 2068.82  4960.7 2066.92
  4987.9 2066.66  4998.3 2065.74  5001.8 2064.73  5002.3 2064.23    5009 2064.73
  5027.7  2066.1  5035.7 2067.65  5049.1 2068.83  5145.2 2068.43  5198.6 2069.11
  5267.1 2071.44  5273.3  2072.5    5292 2072.87  5297.4 2075.17  5316.1 2074.97
  5322.3 2076.54  5327.6 2076.33  5347.2 2078.26  5358.8 2080.98  5422.9 2083.57
#Mann= 3 ,-1 , 0
  4704.1     .07       0  5001.8     .05       0    5009     .07       0
Bank Sta=5001.8,5009
XS Rating Curve= 0 ,0
Exp/Cntr=0.3,0.1

Type RM Length L Ch R = 1 ,23930   ,470,470,470
BEGIN DESCRIPTION:
Rough Hallow 45.0
END DESCRIPTION:
XS GIS Cut Line= 3
      1850074.99     13993474.99        1849975.       13993375.
      1849575.01     13993125.01
#Sta/Elev= 30
  4858.8 2079.66  4887.1  2078.2  4915.4 2074.71  4929.5 2071.88  4943.6 2068.07
  4957.8 2065.51  4986.1 2061.64  5003.2 2062.39  5019.6 2061.49  5020.1 2060.99
  5026.3 2060.99  5026.8 2061.49  5029.1  2063.7  5035.6 2064.53  5050.3 2065.53
  5059.2 2065.41  5117.5 2067.79  5144.7 2067.53  5175.3 2066.43  5188.9 2065.75
  5196.6 2064.27  5202.5 2064.94  5217.8  2064.1    5239 2065.86  5269.7 2065.18
  5283.2  2064.3  5348.7 2067.63  5369.9 2070.13    5443  2077.1  5471.9 2078.15
#Mann= 3 ,-1 , 0
  4858.8     .07       0  5019.6     .05       0  5026.8     .07       0
Bank Sta=5019.6,5026.8
XS Rating Curve= 0 ,0
Exp/Cntr=0.3,0.1

Type RM Length L Ch R = 1 ,23460   ,840,840,840
BEGIN DESCRIPTION:
Rough Hallow 44.0
END DESCRIPTION:
XS GIS Cut Line= 3
        1850425.     13993425.01        1850325.       13993075.
        1849925.       13992675.
#Sta/Elev= 30
    4636 2078.59  4698.4 2078.58  4719.2 2077.14  4730.9 2077.63  4759.5 2075.19
  4764.7 2076.25    4792 2073.05  4798.5 2071.19  4803.7 2072.78  4832.3 2067.73
  4837.5 2069.27    4870 2062.69  4876.5 2062.79  4905.1 2058.83  4910.3 2059.93
  4927.2 2058.32  4944.1 2059.01  4949.3 2058.15  4977.9 2058.17  4993.8 2055.85
  4994.3 2055.35    5001 2055.85  5014.2  2058.6  5028.3 2058.02  5141.4  2061.7
  5183.9 2061.92  5268.7 2060.18    5297 2061.91  5438.4 2066.39  5565.7 2074.31
#Mann= 3 ,-1 , 0
    4636     .07       0  4993.8     .05       0    5001     .07       0
Bank Sta=4993.8,5001
XS Rating Curve= 0 ,0
Exp/Cntr=0.3,0.1

Type RM Length L Ch R = 1 ,22620   ,471,471,471
BEGIN DESCRIPTION:
Rough Hallow 43.0
END DESCRIPTION:
XS GIS Cut Line= 3
      1851225.02     13993175.02        1850225.       13992375.
      1850024.96       13992375.
#Sta/Elev= 30
  3714.3 2070.71  3771.2 2070.23  3806.4 2068.75  3892.8 2067.15  4034.5 2065.97
  4254.6  2062.3  4425.9 2061.84  4475.5  2060.8  4489.9 2058.94  4504.3 2058.37
  4582.8  2059.9  4589.2 2059.31    4618 2059.89  4802.9 2059.42  4909.3 2056.43
  4958.9 2051.81  4981.3 2053.33  4987.8 2052.42    5005 2051.87    5025 2052.01
    5035  2050.5  5035.9  2049.7  5036.4  2049.2    5054  2049.7    5055 2058.25
    5075 2066.26    5085  2068.5    5095 2071.92    5115 2074.81    5195 2077.67
#Mann= 3 ,-1 , 0
  3714.3     .07       0  5035.9     .05       0    5054     .07       0
Bank Sta=5035.9,5054
XS Rating Curve= 0 ,0
Exp/Cntr=0.3,0.1

Type RM Length L Ch R = 1 ,22149   ,480,480,480
BEGIN DESCRIPTION:
Rough Hallow 42.0
END DESCRIPTION:
XS GIS Cut Line= 3
        1851425.       13992875.        1850425.       13991975.
      1850224.96       13991975.
#Sta/Elev= 30
  3654.6 2071.23  3663.4 2071.22  3691.5 2071.16  3739.4  2070.3  3838.8 2066.54
  4058.2 2064.57  4093.7 2063.25  4114.6 2063.72  4348.6 2060.34  4596.4 2055.57
  4603.5 2056.08  4617.7 2054.55  4631.9 2054.26  4702.9 2054.53  4744.7 2052.92
  4758.9 2054.55  4794.8 2055.64  4879.3 2056.51  4929.3 2053.12  4950.3 2054.12
  4971.9 2052.11  4996.6 2046.74  5000.9 2046.65  5001.4 2046.15    5019 2046.65
    5020 2048.14    5050 2062.19    5060 2064.15    5100 2066.54    5200 2069.77
#Mann= 5 ,-1 , 0
  3654.6     .07       0  3663.4      .1       0  3691.5     .07       0
  5000.9     .05       0    5019     .07       0
Bank Sta=5000.9,5019
XS Rating Curve= 0 ,0
Exp/Cntr=0.3,0.1

Type RM Length L Ch R = 1 ,21669   ,861,861,861
BEGIN DESCRIPTION:
Rough Hallow 41.0
END DESCRIPTION:
XS GIS Cut Line= 3
      1851325.01       13991875.      1850761.87     13991682.34
      1850125.03       13991625.
#Sta/Elev= 30
  4409.5 2076.89  4456.5 2073.49  4487.8  2066.3  4494.1 2063.66  4525.8 2056.21
  4550.4 2054.25  4599.8  2052.7  4620.9 2049.98  4644.3 2048.38  4663.2 2048.12
  4694.9 2050.78    4716 2051.17  4795.5 2051.24  4906.3 2053.16    4938 2051.21
  4983.3 2051.82  5000.4 2047.89  5012.4 2046.85  5012.9 2046.35  5030.8 2046.85
  5033.8 2046.95  5051.7 2052.03  5061.8  2051.9  5071.8 2049.68  5091.9 2053.35
  5152.2 2052.77  5192.3 2055.46  5212.4 2055.22  5433.3 2059.72  5644.1 2067.68
#Mann= 3 ,-1 , 0
  4409.5     .07       0  5012.4     .05       0  5030.8     .07       0
Bank Sta=5012.4,5030.8
XS Rating Curve= 0 ,0
Exp/Cntr=0.3,0.1

Type RM Length L Ch R = 1 ,20808   ,443,443,443
BEGIN DESCRIPTION:
Rough Hallow 40.0
END DESCRIPTION:
XS GIS Cut Line= 3
      1851224.95     13991025.01        1851025.       13991075.
        1849925.       13991675.
#Sta/Elev= 30
  4789.3 2079.93  4807.3 2078.07  4820.2 2073.92  4848.5 2072.55  4853.7    2071
    4931 2063.77  4936.1 2062.45  4954.2 2053.77  4964.5 2047.65  4983.6 2040.39
  4984.1 2039.89  5002.1 2040.39  5025.3 2042.43    5031 2044.59  5063.3 2046.19
  5106.9 2044.63  5112.6 2042.72  5143.5 2045.84  5166.3 2046.87  5194.3 2047.78
  5210.4 2046.92    5246 2049.06  5275.9  2048.6  5348.5 2051.72  5651.8 2053.77
  5815.1 2056.96  5924.2  2062.7  6055.2 2067.85  6145.9 2073.52  6248.4 2075.95
#Mann= 3 ,-1 , 0
  4789.3     .07       0  4983.6     .05       0  5002.1     .07       0
Bank Sta=4983.6,5002.1
XS Rating Curve= 0 ,0
Exp/Cntr=0.3,0.1

Type RM Length L Ch R = 1 ,20365   ,371,371,371
BEGIN DESCRIPTION:
Rough Hallow 39.0
END DESCRIPTION:
XS GIS Cut Line= 3
        1850975.       13990675.        1850775.       13990725.
      1849774.99       13991225.
#Sta/Elev= 30
  4794.1 2071.15  4853.4  2065.7  4917.8 2062.27  4948.7 2054.73  4982.2 2049.73
  4997.7 2044.76  5003.1 2044.76  5014.2 2040.18  5053.4 2043.17  5067.3 2043.16
  5098.1 2042.46  5120.4 2039.84    5126 2041.77  5148.4 2043.05  5165.2 2042.86
  5179.1 2039.66  5200.6 2038.27  5201.1 2037.77  5219.1 2038.27  5223.9 2040.93
  5232.3 2040.31  5260.2 2042.92  5299.3 2042.22  5394.4 2046.16  5545.3 2046.94
  5701.8 2051.82  5768.9 2056.53    5850 2059.43  6020.5 2069.08  6118.3  2072.2
#Mann= 3 ,-1 , 0
  4794.1     .07       0  5200.6     .05       0  5219.1     .07       0
Bank Sta=5200.6,5219.1
XS Rating Curve= 0 ,0
Exp/Cntr=0.3,0.1

Type RM Length L Ch R = 1 ,19994   ,547,547,547
BEGIN DESCRIPTION:
Rough Hallow 38.0
END DESCRIPTION:
XS GIS Cut Line= 3
      1850974.97     13990275.02      1850477.18      13990549.3
      1849824.98     13991125.01
#Sta/Elev= 30
  4447.7 2080.57  4542.8 2073.26  4580.7 2068.06  4624.2 2065.59  4705.6 2058.82
  4933.8 2051.39  4949.8 2049.58  4955.5 2046.03  4971.6 2042.62  4977.3 2038.13
  4993.4 2038.32  5035.6 2042.15  5078.3 2042.22  5113.4 2040.09  5141.8 2040.18
  5156.1 2038.32  5163.6 2038.55  5175.3 2035.79  5175.8 2035.29  5193.8 2035.79
  5198.7 2037.78  5205.7 2038.36  5219.6 2037.92  5233.9 2040.09    5305  2043.3
  5439.7 2044.79    5525 2046.91  5666.4  2058.6  5815.3 2064.59    5886 2069.07
#Mann= 3 ,-1 , 0
  4447.7     .07       0  5175.3     .05       0  5193.8     .07       0
Bank Sta=5175.3,5193.8
XS Rating Curve= 0 ,0
Exp/Cntr=0.3,0.1

Type RM Length L Ch R = 1 ,19447   ,463,463,463
BEGIN DESCRIPTION:
Rough Hallow 37.0
END DESCRIPTION:
XS GIS Cut Line= 3
      1850625.02     13990224.99        1850025.       13990525.
        1849775.       13990775.
#Sta/Elev= 30
    4333 2056.02  4369.4 2054.55  4609.7 2048.74  4683.8 2047.91  4704.8 2047.32
  4721.5 2045.89  4727.1 2044.41  4743.9 2043.37  4749.9 2041.47  4816.6 2036.56
  4869.7    2039    4892 2037.51  4900.4 2037.87  4914.4  2036.4  4936.8 2035.98
  4945.1 2037.42  4967.5 2037.08  4989.9 2034.48  4991.8 2033.35  4992.3 2032.85
  5010.4 2033.35    5018 2040.43  5074.6 2042.28  5131.1 2042.22  5201.8 2043.13
  5230.1 2044.23  5258.4 2047.95  5300.8 2055.43  5329.1 2058.47  5357.4 2059.68
#Mann= 5 ,-1 , 0
    4333     .07       0  4683.8    .035       0  4749.9     .07       0
  4991.8     .05       0  5010.4     .07       0
Bank Sta=4991.8,5010.4
XS Rating Curve= 0 ,0
Exp/Cntr=0.3,0.1

Type RM Length L Ch R = 1 ,18984   ,515,515,515
BEGIN DESCRIPTION:
Rough Hallow 36.1
END DESCRIPTION:
XS GIS Cut Line= 4
      1850818.72     13989887.71      1850128.34     13990092.27
      1849699.07     13990103.08       1849070.3     13990121.54
#Sta/Elev= 30
  4076.1 2078.51  4111.3 2077.11  4173.8  2069.2  4256.1 2063.91  4351.2 2053.59
  4471.2 2048.43  4685.1 2042.21  4752.8 2039.07    4789 2039.68  4939.5 2037.04
  4959.5 2029.94  4979.5 2028.94  4989.6 2028.87  5009.6 2033.47  5039.6 2034.76
  5049.6 2033.39  5050.2 2028.39  5050.7 2027.89  5068.9 2028.39  5069.6 2030.07
  5079.6 2031.69  5109.6 2033.22  5119.6 2037.52  5159.6 2047.82  5199.6 2050.84
  5269.6 2053.21  5309.7  2056.9  5429.7 2063.41  5629.8 2068.12  5854.6 2076.09
#Mann= 5 ,-1 , 0
  4076.1     .07       0  4685.1    .035       0    4789     .07       0
  5050.2     .05       0  5068.9     .07       0
Bank Sta=5050.2,5068.9
XS Rating Curve= 0 ,0
Exp/Cntr=0.3,0.1

Type RM Length L Ch R = 1 ,18469   ,467,467,467
BEGIN DESCRIPTION:
Rough Hallow 36.0
END DESCRIPTION:
XS GIS Cut Line= 3
      1850475.05       13989725.        1850275.       13989725.
      1849079.31     13989660.04
#Sta/Elev= 30
  4795.8 2049.86  4865.8 2046.81  4925.8 2040.92  4965.8  2033.3  4985.8 2027.62
  4993.3 2024.32  4995.8 2024.32  4996.5 2023.35    4997 2022.85  5015.3 2023.35
  5025.9 2025.19  5035.9 2024.89    5076 2028.44  5084.5 2031.08    5096 2031.04
    5126 2033.88  5176.1 2036.63  5216.2 2037.53  5306.3 2042.07  5326.3 2044.19
  5396.4  2047.2  5486.6 2049.76  5496.6 2050.81  5596.7  2052.5  5636.4 2054.56
  5736.9 2057.23  5828.7 2058.47  6011.1 2064.92  6037.4 2066.73  6193.3 2070.28
#Mann= 4 ,-1 , 0
  4795.8     .07       0  4996.5     .05       0  5015.3     .07       0
  6011.1      .1       0
Bank Sta=4996.5,5015.3
XS Rating Curve= 0 ,0
Exp/Cntr=0.3,0.1

Type RM Length L Ch R = 1 ,18002   ,482,482,482
BEGIN DESCRIPTION:
Rough Hallow 35.0
END DESCRIPTION:
XS GIS Cut Line= 3
      1850525.02     13989325.01        1850325.       13989275.
      1849409.48     13989288.78
#Sta/Elev= 30
  4793.9 2057.72  4835.2 2054.95  4845.5 2054.89  4853.2 2053.24  4876.4 2050.55
  4927.9 2047.88  4935.7 2046.15  4940.8 2046.14  4969.2 2038.95  4976.9 2036.21
    4982 2035.77  4997.5 2027.36  5002.6 2027.36  5010.1 2023.11  5010.7 2021.69
  5011.2 2021.19  5029.5 2021.69  5030.1  2023.9  5060.1 2025.45  5070.1 2027.99
  5130.1  2028.9  5250.1 2037.77  5290.1 2038.34  5360.1 2041.55  5380.1 2043.15
  5500.1 2045.76  5600.1 2049.01  5770.2 2052.65  5840.2 2054.95  5915.7 2056.25
#Mann= 3 ,-1 , 0
  4793.9     .07       0  5010.7     .05       0  5029.5     .07       0
Bank Sta=5010.7,5029.5
XS Rating Curve= 0 ,0
Exp/Cntr=0.3,0.1

Type RM Length L Ch R = 1 ,17520   ,461,461,461
BEGIN DESCRIPTION:
Rough Hallow 34.0
END DESCRIPTION:
XS GIS Cut Line= 3
      1850425.01       13988775.        1850225.       13988825.
      1849824.97     13989075.02
#Sta/Elev= 30
  4802.2 2049.66  4843.4 2047.14  4884.7 2042.09  4925.9 2033.72  4943.9 2028.34
  4949.1 2028.34  4956.8 2025.55  4975.7 2023.23  4976.2 2022.73  4994.1 2022.73
  4994.6 2023.23  5005.8 2026.42  5037.3 2026.33  5043.7 2024.96  5067.3 2024.09
    5095 2025.32  5102.7 2026.99  5110.4 2027.66  5116.3 2027.39  5131.6 2028.14
  5146.9  2030.4  5152.8 2029.93  5168.2    2031  5174.1 2030.41    5197 2032.14
  5268.4 2034.87    5305 2037.47  5356.8 2039.28  5421.1 2042.56  5480.1 2043.99
#Mann= 3 ,-1 , 0
  4802.2     .07       0  4975.7     .05       0  4994.6     .07       0
Bank Sta=4975.7,4994.6
XS Rating Curve= 0 ,0
Exp/Cntr=0.3,0.1

Type RM Length L Ch R = 1 ,17059   ,450,450,450
BEGIN DESCRIPTION:
Rough Hallow 33.0
END DESCRIPTION:
XS GIS Cut Line= 3
      1850424.98       13988475.        1850125.       13988425.
      1849775.03     13988624.98
#Sta/Elev= 30
  4700.1 2049.16    4733 2046.07  4760.9 2042.44  4788.8 2037.66  4793.9 2037.65
  4821.7 2032.43  4849.6  2025.7  4854.7 2025.73  4862.3 2024.21  4882.6 2022.89
  4892.7 2023.81  4943.4 2022.62  4963.7 2023.74  4971.3 2023.48  4974.5 2021.96
    4975 2021.46  4992.9 2021.46  4993.4 2021.96  5001.7 2023.41  5027.3 2024.83
  5033.7 2026.01  5055.3 2027.79  5071.2 2030.03  5130.2 2032.05  5246.1 2034.22
  5297.2 2037.38  5318.8 2039.65  5356.2 2041.47  5377.8 2041.36  5407.3 2042.38
#Mann= 3 ,-1 , 0
  4700.1     .07       0  4974.5     .05       0  4993.4     .07       0
Bank Sta=4974.5,4993.4
XS Rating Curve= 0 ,0
Exp/Cntr=0.3,0.1

Type RM Length L Ch R = 1 ,16609   ,445,445,445
BEGIN DESCRIPTION:
Rough Hallow 32.0
END DESCRIPTION:
XS GIS Cut Line= 3
      1850324.99       13987975.        1850075.       13988025.
      1849336.53     13988390.48
#Sta/Elev= 30
  4749.9 2041.27  4790.7 2038.97  4821.3 2035.98  4831.5 2033.83  4851.9 2031.52
  4862.1 2029.35  4882.5 2022.29  4892.7 2020.91  4964.8 2019.45  4965.3 2018.95
  4983.2 2018.95  4983.7 2019.45  4984.4 2020.34  4994.6 2019.78  5002.3 2020.55
  5007.6 2020.55  5013.3 2022.06  5108.6 2026.39  5138.7 2028.59    5260 2033.72
  5377.7 2036.53  5451.2 2037.78  5562.7 2040.94  5585.2 2041.16  5607.6 2042.18
  5669.3  2043.6  5685.5 2044.43  5719.8 2044.69  5781.5 2046.31  5828.8 2048.06
#Mann= 3 ,-1 , 0
  4749.9     .07       0  4964.8     .05       0  4983.7     .07       0
Bank Sta=4964.8,4983.7
XS Rating Curve= 0 ,0
Exp/Cntr=0.3,0.1

Type RM Length L Ch R = 1 ,16164   ,618,618,618
BEGIN DESCRIPTION:
Rough Hallow 31.0
END DESCRIPTION:
XS GIS Cut Line= 4
      1850274.95     13987674.99        1850025.       13987625.
        1849625.       13987875.      1849219.81     13988169.13
#Sta/Elev= 30
  4750.8 2036.69  4801.7 2034.97  4852.7 2031.79  4883.3  2029.2  4913.9 2024.59
  4934.3 2022.89  4954.7 2020.29  4964.9 2017.13  4975.1 2015.55  4985.3 2014.51
  4993.7 2014.49  4994.2 2013.99  5012.1 2013.99  5012.6 2014.49  5013.4 2015.13
  5071.2 2021.13  5113.6 2022.28  5144.3 2024.43  5171.4 2025.37    5202 2025.04
  5223.3 2025.74  5281.1 2028.39  5317.6 2030.83  5360.1 2032.23    5412 2033.23
    5442 2034.59  5541.2 2035.76  5555.9 2036.65  5671.1 2037.93  5978.1 2044.71
#Mann= 3 ,-1 , 0
  4750.8     .07       0  4993.7     .05       0  5012.6     .07       0
Bank Sta=4993.7,5012.6
XS Rating Curve= 0 ,0
Exp/Cntr=0.3,0.1

Type RM Length L Ch R = 1 ,15546   ,486,486,486
BEGIN DESCRIPTION:
Rough Hallow 30.1
END DESCRIPTION:
XS GIS Cut Line= 4
      1850642.24     13987103.37      1849996.57     13987039.37
      1849610.21     13987137.11      1849215.56     13987156.76
#Sta/Elev= 30
  4173.7 2036.42  4271.4 2034.51  4281.5  2035.1  4312.9 2034.13    4603 2031.54
    4804 2020.24  4827.2 2019.58  4855.1 2015.82    4917 2015.09  4927.3 2013.71
  4937.6 2011.16  4945.1  2012.1  4950.3 2011.74  4958.2 2014.13  4968.6 2013.53
  4975.5 2010.64    4976 2010.14  4996.7 2010.64  4999.5 2013.64  5027.1 2023.32
  5032.3 2023.11  5040.8 2024.79  5068.2 2027.07    5082 2027.41  5109.2 2029.98
  5114.3 2029.43  5133.6  2031.4  5296.4 2038.76  5475.9 2048.89  5616.2 2054.89
#Mann= 3 ,-1 , 0
  4173.7     .07       0  4975.5     .05       0  4996.7     .07       0
Bank Sta=4975.5,4996.7
XS Rating Curve= 0 ,0
Exp/Cntr=0.3,0.1

Type RM Length L Ch R = 1 ,15060   ,488,488,488
BEGIN DESCRIPTION:
Rough Hallow 30.0
END DESCRIPTION:
XS GIS Cut Line= 3
      1850422.54     13986820.43        1849825.       13986625.
        1849475.       13986425.
#Sta/Elev= 30
  4379.7 2032.58  4398.2 2033.41  4419.2 2032.42  4578.2 2031.99  4598.1 2030.55
  4641.9 2029.57  4668.5 2027.55  4673.8 2028.06  4764.1 2023.52  4801.3 2019.58
    4819 2014.98  4850.6 2011.34  4903.2 2014.89  4923.5    2012  4924.1 2011.18
  4924.6 2010.68  4945.3 2011.18  4955.3 2015.66  4976.8 2015.01  4997.9 2011.57
  5011.3  2012.3  5022.1 2014.71  5037.9 2027.89  5053.7  2031.6    5112 2038.31
  5118.5  2039.8  5140.1 2041.25  5177.6 2046.03  5285.5 2053.05  5411.5 2058.07
#Mann= 3 ,-1 , 0
  4379.7     .07       0  4924.1     .05       0  4945.3     .07       0
Bank Sta=4924.1,4945.3
XS Rating Curve= 0 ,0
Exp/Cntr=0.3,0.1

Type RM Length L Ch R = 1 ,14572   ,575,575,575
BEGIN DESCRIPTION:
Rough Hallow 29.0
END DESCRIPTION:
XS GIS Cut Line= 4
      1850325.02     13986725.04      1850109.97     13986251.93
      1850000.33     13986184.33      1849674.96     13986225.01
#Sta/Elev= 30
  4398.9 2032.25  4436.3 2032.44  4453.9 2031.42  4551.6  2030.3  4557.1 2030.84
  4640.6 2026.92  4706.5 2022.49  4761.4 2021.55  4844.9 2014.02  4850.4 2012.08
  4896.5 2009.54  4935.8 2011.35    4963 2010.52  4984.2 2008.74    4989 2006.89
  4989.5 2006.39  5010.2 2006.89  5030.2 2012.03  5036.3 2018.04    5042 2020.57
  5047.4 2020.57  5052.8 2024.68  5090.6 2034.42  5095.6 2033.48  5133.4 2038.22
  5171.2 2040.91    5214 2043.23  5256.8 2044.34  5324.9 2048.68  5375.3  2050.8
#Mann= 3 ,-1 , 0
  4398.9     .07       0    4989     .05       0  5010.2     .07       0
Bank Sta=4989,5010.2
XS Rating Curve= 0 ,0
Exp/Cntr=0.3,0.1

Type RM Length L Ch R = 1 ,13997   ,585,585,585
BEGIN DESCRIPTION:
Rough Hallow 28.0
END DESCRIPTION:
XS GIS Cut Line= 3
      1850793.42     13986371.48      1850384.62     13985766.71
      1850025.01       13985725.
#Sta/Elev= 30
  4268.8 2029.63  4409.4 2026.75  4445.6 2024.65  4596.4 2021.67  4647.3 2019.87
  4761.3 2018.83  4833.2 2014.05  4842.1    2013  4848.1 2011.21  4863.1 2010.01
  4869.1 2008.66  4878.1 2008.27  4899.1 2009.72  4920.1 2008.95    4935 2009.62
    4950  2008.3    4971  2004.9  5007.9 2003.95  5008.4 2003.45  5029.2 2003.95
  5038.7 2008.05  5048.7 2009.78  5060.4 2013.82  5078.9 2017.23    5089 2018.22
  5129.3 2020.78  5159.5 2023.72  5189.7  2024.9    5240 2028.41  5360.8 2034.01
#Mann= 3 ,-1 , 0
  4268.8     .07       0  5007.9     .05       0  5029.2     .07       0
Bank Sta=5007.9,5029.2
XS Rating Curve= 0 ,0
Exp/Cntr=0.3,0.1

Type RM Length L Ch R = 1 ,13412   ,571,571,571
BEGIN DESCRIPTION:
Rough Hallow 27.0
END DESCRIPTION:
XS GIS Cut Line= 4
      1851125.02     13985675.02      1850928.29      13985445.5
      1850706.64       13985325.      1850175.02       13985325.
#Sta/Elev= 30
  4532.2 2036.47  4704.7 2028.72  4744.6 2026.45  4766.6 2026.14  4808.8 2022.36
  4815.9 2022.48  4830.2 2020.33  4833.2  2018.1  4839.2  2018.1  4850.7 2013.21
    4861 2011.17  4866.8 2009.05  4895.1  2005.7  4899.6 2003.67  4900.1 2003.17
  4921.4 2003.67  4932.4 2005.25  4940.7 2004.66  4950.3 2005.53  4976.1 2005.76
  4997.9 2004.85  5035.9 2006.41  5043.1 2007.44  5073.9 2006.57  5090.1 2007.49
  5158.4 2014.59  5318.4 2021.94  5338.4 2021.99  5418.4 2025.85  5618.4 2029.78
#Mann= 5 ,-1 , 0
  4532.2     .07       0  4704.7    .035       0  4899.6     .05       0
  4921.4    .035       0  4950.3     .07       0
Bank Sta=4899.6,4921.4
XS Rating Curve= 0 ,0
Exp/Cntr=0.3,0.1

Type RM Length L Ch R = 1 ,12841   ,246,246,246
BEGIN DESCRIPTION:
Rough Hallow 26.0
END DESCRIPTION:
XS GIS Cut Line= 3
      1851375.02     13985175.01        1851025.       13984975.
      1850425.01       13985075.
#Sta/Elev= 30
  4601.2 2038.65  4829.4 2031.42  4866.1 2031.27  4872.6 2029.99  4894.2 2029.49
  4915.8 2027.51  4923.7 2024.97  4931.6 2020.89  4937.4 2021.38  4946.7 2009.81
  4953.2 2003.52    4959 2002.67  4969.1 1999.45  4981.3 1999.38  4990.6 1998.28
  4991.1 1997.78  5011.9 1997.78  5012.4 1998.28  5014.5 1999.38  5037.3 1999.35
  5044.9 2001.09  5075.3 2003.93  5166.5 2009.15  5280.6  2010.6  5298.3 2012.46
  5308.5 2012.44    5352 2014.87  5430.1 2020.06  5551.8 2022.06  5612.6 2023.97
#Mann= 4 ,-1 , 0
  4601.2     .07       0  4990.6     .05       0  5012.4     .07       0
    5352    .035       0
Bank Sta=4990.6,5012.4
XS Rating Curve= 0 ,0
Exp/Cntr=0.3,0.1

Type RM Length L Ch R = 1 ,12595   ,280,280,280
BEGIN DESCRIPTION:
Mapping XS 41deb7da
END DESCRIPTION:
XS GIS Cut Line= 2
      1851670.29     13984553.28       1850322.9     13985045.83
#Sta/Elev= 30
    4367 2031.63  4457.8 2028.27  4479.2 2026.32  4574.9  2022.2  4660.1 2012.51
  4702.2  2010.3  4732.7 2007.39    4738 2007.72  4768.6 2016.03  4793.8 2017.21
  4824.3  2020.6  4915.9  2022.8  4971.6  2021.6  4979.5 2019.17  4996.9 2001.91
  5002.2 2002.21  5016.4 1998.32  5016.9 1997.82  5038.3 1998.32  5043.4 2000.23
  5057.9 1999.35  5064.7 2001.16  5075.4 2000.58  5144.2 2002.81  5181.8 2007.76
  5213.8 2009.05  5322.1 2010.73  5543.8 2021.16    5661 2022.67  5801.6 2026.45
#Mann= 3 ,-1 , 0
    4367     .07       0  5016.4     .05       0  5038.3     .07       0
Bank Sta=5016.4,5038.3
XS Rating Curve= 0 ,0
Exp/Cntr=0.3,0.1

Type RM Length L Ch R = 1 ,12315   ,571,571,571
BEGIN DESCRIPTION:
Rough Hallow 25.0
END DESCRIPTION:
XS GIS Cut Line= 3
      1851432.06     13984346.55        1850975.       13984525.
      1850258.36     13984751.05
#Sta/Elev= 30
  4509.6 2031.36  4537.6 2028.75  4613.2 2025.16  4678.2 2022.95  4752.1 2018.13
  4822.3 2008.79  4846.8 2003.41  4852.2 2005.62    4863 2001.74  4871.3 2000.15
  4876.7 2003.52  4906.5 2002.55  4914.4 2000.75  4955.5 2002.08  4966.5 2000.87
  4978.8 2000.32  4979.4 1999.25  4979.9 1998.75    5002 1999.25  5016.4 2000.29
  5042.2 1999.56  5071.9 2001.55  5133.8    2009  5151.1 2008.21  5199.5 2009.35
  5385.3 2015.28  5430.4 2016.37  5524.5 2019.18  5646.9 2019.93  5751.7 2022.01
#Mann= 13 ,-1 , 0
  4509.6    .035       0  4537.6     .07       0  4613.2    .035       0
  4752.1     .07       0    4863    .063       0  4966.5     .07       0
  4979.4     .05       0    5002     .07       0  5071.9     .07       0
  5133.8    .035       0  5385.3      .1       0  5430.4    .063       0
  5646.9     .07       0
Bank Sta=4979.4,5002
XS Rating Curve= 0 ,0
Exp/Cntr=0.3,0.1

Type RM Length L Ch R = 1 ,11744   ,558,558,558
BEGIN DESCRIPTION:
Rough Hallow 24.0
END DESCRIPTION:
XS GIS Cut Line= 3
      1850875.01     13983724.98        1850675.       13984075.
      1850575.01     13984474.96
#Sta/Elev= 30
  4596.9 2043.07  4610.6 2041.91  4654.5 2041.37  4735.1 2037.12  4750.2 2035.44
  4758.2 2036.29  4793.4 2032.61  4815.8 2032.08  4852.5 2029.19  4868.3 2029.39
  4905.7 2026.72  4927.3 2023.39  4933.1 2021.47  4942.4 2016.88  4964.8 2003.54
    4977 1992.41  4980.8 1987.63  4981.3 1987.13  5003.4 1987.63    5031  1993.5
  5072.2  1996.6  5082.5  1996.9  5092.8 1995.33  5100.5 1996.87    5134  1999.7
    5183 2005.24  5278.3 2008.39    5299 2010.01  5353.1 2012.15  5412.3 2013.81
#Mann= 3 ,-1 , 0
  4596.9      .1       0  4980.8     .05       0  5003.4      .1       0
Bank Sta=4980.8,5003.4
XS Rating Curve= 0 ,0
Exp/Cntr=0.3,0.1

Type RM Length L Ch R = 1 ,11186   ,559,559,559
BEGIN DESCRIPTION:
Rough Hallow 23.0
END DESCRIPTION:
XS GIS Cut Line= 3
      1850624.98     13983675.01        1850225.       13983775.
        1850025.       13984125.
#Sta/Elev= 30
  4583.1 2034.35  4642.3 2029.37    4730 2024.38  4758.3 2021.88  4799.5 2016.91
    4815 2012.98  4875.9 2003.06  4923.2 1998.46    4931  1996.4  4943.8 1991.12
  4954.2 1988.57  4978.4 1987.52  4985.1 1988.31  4997.8  1986.9  4998.3  1986.4
  5020.4  1986.9  5024.9 1991.41  5030.7 1991.87  5046.5    1997    5053 1997.68
  5105.5 1998.75  5111.3 1997.76  5121.4 1998.13  5127.1 1997.29  5164.6 2001.16
  5171.2 2001.15  5186.1 2003.21  5245.2 2008.35  5363.2 2015.65  5398.5 2017.09
#Mann= 6 ,-1 , 0
  4583.1      .1       0  4875.9     .07       0  4978.4     .07       0
  4997.8     .05       0  5020.4     .07       0  5171.2      .1       0
Bank Sta=4997.8,5020.4
XS Rating Curve= 0 ,0
Exp/Cntr=0.3,0.1

Type RM Length L Ch R = 1 ,10627   ,533,533,533
BEGIN DESCRIPTION:
Rough Hallow 22.0
END DESCRIPTION:
XS GIS Cut Line= 3
      1850124.99     13983175.01        1849775.       13983475.
      1849574.99     13983825.02
#Sta/Elev= 30
  4544.3 2019.08  4586.5 2016.26  4657.9 2010.02  4664.5 2010.16  4756.7 2002.13
  4764.4 2002.55    4828 1999.21  4926.8 1995.45    4963  1990.2  4977.3 1987.14
  4980.2 1984.33  4980.7 1983.83  5002.9 1984.33  5005.3  1987.1  5013.2 1987.61
  5050.6 1987.48  5056.4 1985.68  5062.9 1987.52  5085.9 1988.59  5099.6 1986.73
  5108.9 1989.51  5115.4 1994.11  5121.2 2001.11    5137 2006.91  5210.2 2012.75
  5221.5 2013.52  5292.5 2018.32  5357.3 2020.37  5378.9 2020.09  5408.4 2021.54
#Mann= 5 ,-1 , 0
  4544.3      .1       0  4980.2     .05       0  5002.9      .1       0
  5210.2     .07       0  5221.5      .1       0
Bank Sta=4980.2,5002.9
XS Rating Curve= 0 ,0
Exp/Cntr=0.3,0.1

Type RM Length L Ch R = 1 ,10094   ,547,547,547
BEGIN DESCRIPTION:
Rough Hallow 21.0
END DESCRIPTION:
XS GIS Cut Line= 3
      1849924.96     13982825.02        1849425.       13983125.
      1849224.98     13983475.03
#Sta/Elev= 30
  4411.2 2019.67  4446.1 2017.46  4477.2  2013.5  4514.2 2010.49  4551.1 2008.66
  4621.1 2003.47  4827.1 1995.37  4842.6 1993.94    4864  1989.6  4877.6 1987.82
    4901 1987.82  4928.2 1986.54  4949.5  1983.5  4970.9 1983.37  4994.2 1980.11
  4996.5 1977.99    4997 1977.49  5019.3 1977.99  5023.8 1980.13  5029.5 1986.31
  5039.6 1991.65  5045.4 2000.97    5067 2005.18  5097.9 2007.85  5110.1 2009.71
  5120.2 2008.97  5200.8 2011.34  5299.3 2015.54  5322.1 2016.26  5397.4  2017.6
#Mann= 5 ,-1 , 0
  4411.2      .1       0  4996.5     .05       0  5019.3      .1       0
  5299.3     .07       0  5322.1      .1       0
Bank Sta=4996.5,5019.3
XS Rating Curve= 0 ,0
Exp/Cntr=0.3,0.1

Type RM Length L Ch R = 1 ,9547    ,439,439,439
BEGIN DESCRIPTION:
Rough Hallow 20.0
END DESCRIPTION:
XS GIS Cut Line= 3
      1849625.04     13982324.97        1849175.       13982675.
      1848975.02     13983024.96
#Sta/Elev= 30
  4434.4 2017.16    4591  2006.1  4640.8 2003.37  4662.5 2001.04  4748.4 1997.65
  4790.1  1993.1  4804.5 1990.84  4827.2 1985.81  4839.8 1984.67  4862.5 1985.63
  4912.2 1979.35  4930.4 1982.01  4943.6 1982.26  4953.9  1982.4  4968.3 1980.52
  4976.5 1980.38  4979.6 1977.01  4980.1 1976.51  5002.4 1977.01  5012.5 1979.15
  5018.2  1984.5  5027.6    1986    5034 1988.17  5039.8  1991.6  5049.9 1993.18
  5055.6 1995.55  5062.1 1996.91  5079.6 1999.32  5152.1 2003.25  5407.6 2011.73
#Mann= 6 ,-1 , 0
  4434.4      .1       0  4930.4     .07       0  4943.6      .1       0
  4979.6     .05       0  5002.4      .1       0  5079.6     .07       0
Bank Sta=4979.6,5002.4
XS Rating Curve= 0 ,0
Exp/Cntr=0.3,0.1

Type RM Length L Ch R = 1 ,9108    ,177,177,177
BEGIN DESCRIPTION:
Rough Hallow 19.1
END DESCRIPTION:
XS GIS Cut Line= 2
      1849441.77     13981857.34      1848869.09     13982607.66
#Sta/Elev= 30
  4471.9 2016.76  4481.3 2015.55  4516.3 2013.53  4602.1 2008.58  4686.1 2002.96
  4722.8 1999.11    4739 1998.23  4753.5 1992.09    4768 1990.59  4843.5  1988.1
  4855.8 1989.08  4874.1 1988.53  4882.3 1990.04  4888.6 1988.76  4903.2 1991.32
  4909.5 1989.09  4946.8 1986.83  4964.3 1982.56  4991.5  1977.4    4992  1976.9
  5014.3  1977.4  5088.2 1980.44  5123.5 1978.15  5181.6 1985.59  5187.9 1987.91
  5237.8 1995.73  5274.1 1999.67  5326.4 2001.09  5365.1 2002.22  5415.8 2003.51
#Mann= 13 ,-1 , 0
  4471.9     .07       0  4481.3      .1       0  4516.3    .063       0
  4602.1    .035       0  4686.1    .063       0  4722.8    .035       0
  4843.5      .1       0  4855.8    .063       0  4964.3     .07       0
  4991.5     .05       0  5014.3     .07       0  5326.4     .07       0
  5365.1    .035       0
Bank Sta=4991.5,5014.3
XS Rating Curve= 0 ,0
Exp/Cntr=0.3,0.1

Type RM Length L Ch R = 1 ,8931    ,469,469,469
BEGIN DESCRIPTION:
Rough Hallow 19.0
END DESCRIPTION:
XS GIS Cut Line= 3
      1849280.83     13981796.66      1849031.97     13982130.98
      1848775.25     13982483.42
#Sta/Elev= 30
  4582.8 2018.95  4779.6 2010.49  4785.8 2011.54  4800.4  2009.5  4806.6 2010.52
    4815 2008.82  4850.5 2007.71  4860.8 2006.25  4885.9 2005.05  4899.1 2002.54
    4936 1997.58  4942.3 1994.42  4965.2    1988  4971.4 1984.49  4992.2 1976.15
  5015.3 1975.03  5017.8 1973.85  5018.3 1973.35  5040.8 1973.85  5042.4 1975.95
  5050.9 1977.14  5071.7 1978.41  5115.8 1978.84  5121.9 1980.45  5128.3 1979.97
  5157.5 1981.82    5193 1987.62  5278.8 1996.34  5379.2  2002.3  5435.6 2002.43
#Mann= 5 ,-1 , 0
  4582.8    .035       0  4860.8      .1       0  4899.1     .07       0
  5017.8     .05       0  5040.8     .07       0
Bank Sta=5017.8,5040.8
XS Rating Curve= 0 ,0
Exp/Cntr=0.3,0.1

Type RM Length L Ch R = 1 ,8462    ,564,564,564
BEGIN DESCRIPTION:
Rough Hallow 18.0
END DESCRIPTION:
XS GIS Cut Line= 3
      1848874.98     13981525.03        1848675.       13981875.
        1848575.     13982275.01
#Sta/Elev= 30
  4601.5 2023.72  4739.7 2019.69  4762.7 2019.92  4820.3 2017.33  4829.7 2017.61
  4835.4 2016.16  4866.4 2013.35  4897.6 2008.88  4910.3 2005.72    4916 2003.57
  4937.6 1991.39    4947 1977.58  4969.3  1970.6  4981.5 1970.56  5003.4 1968.73
  5003.9 1968.23  5026.4 1968.73  5027.8 1972.17    5069  1975.5  5078.1 1977.61
    5087  1979.8  5097.3 1980.18    5118 1983.67  5159.2  1986.8  5187.5 1988.47
    5221 1988.52  5303.5 1992.46  5352.5 1997.18    5386 1998.15  5416.9 2000.29
#Mann= 5 ,-1 , 0
  4601.5      .1       0  4897.6     .07       0  5003.4     .05       0
  5026.4     .07       0  5078.1      .1       0
Bank Sta=5003.4,5026.4
XS Rating Curve= 0 ,0
Exp/Cntr=0.3,0.1

Type RM Length L Ch R = 1 ,7898    ,567,567,567
BEGIN DESCRIPTION:
Rough Hallow 17.0
END DESCRIPTION:
XS GIS Cut Line= 3
      1848524.98     13981475.01        1848175.       13981675.
        1848225.       13982075.
#Sta/Elev= 30
  4597.9 2015.35  4655.5  2014.8  4701.5 2011.91  4723.8 2012.29  4862.8 2007.06
  4885.1 2004.82  4890.9 2002.29  4906.7  2000.3  4910.5 1997.75  4928.3 1993.67
    4934 1989.93  4949.9 1988.14  4955.6 1978.95  4965.7 1978.44  4971.5 1969.35
  4993.1 1959.61  4999.5 1959.25    5000 1958.75  5022.6 1959.25  5038.8 1963.94
  5043.8 1963.04  5049.8 1965.97  5071.5 1971.38  5124.4 1973.43  5162.2 1976.99
  5212.6  1984.1  5252.9 1984.21  5309.2 1986.89  5345.5 1989.27  5404.1 1991.81
#Mann= 7 ,-1 , 0
  4597.9      .1       0  4910.5     .07       0  4999.5     .05       0
  5022.6     .07       0  5049.8      .1       0  5309.2     .07       0
  5345.5      .1       0
Bank Sta=4999.5,5022.6
XS Rating Curve= 0 ,0
Exp/Cntr=0.3,0.1

Type RM Length L Ch R = 1 ,7331    ,563,563,563
BEGIN DESCRIPTION:
Rough Hallow 16.0
END DESCRIPTION:
XS GIS Cut Line= 3
      1847825.02     13981274.97        1847625.       13981625.
        1847625.     13982024.95
#Sta/Elev= 30
  4596.5 2001.76  4677.2 1999.87  4803.1 1991.75  4861.4 1984.36  4869.3  1981.9
  4889.5 1977.43    4896 1974.93    4919 1972.32  4926.9  1968.2  4942.1 1964.78
  4948.5 1962.07  4952.6 1957.85  4953.1 1957.35  4976.1 1957.85  4976.6 1959.27
  4991.7 1959.56  5019.6 1958.61  5031.7 1962.05  5039.6 1964.95  5049.6 1965.09
  5059.6 1966.76  5069.6 1970.17  5099.6 1972.87  5129.6 1982.45  5139.6 1983.23
  5149.6 1985.79  5179.6 1989.66  5299.6    1994  5319.6 1995.72  5399.6 1997.72
#Mann= 5 ,-1 , 0
  4596.5      .1       0  4869.3     .07       0  4952.6     .05       0
  4976.1     .07       0  5031.7      .1       0
Bank Sta=4952.6,4976.1
XS Rating Curve= 0 ,0
Exp/Cntr=0.3,0.1

Type RM Length L Ch R = 1 ,6768    ,544,544,544
BEGIN DESCRIPTION:
Rough Hallow 15.0
END DESCRIPTION:
XS GIS Cut Line= 3
      1847324.99     13981175.01        1847125.       13981525.
      1846925.01     13981874.99
#Sta/Elev= 30
    4597 1990.13  4707.1 1983.24  4712.9 1983.66  4787.7 1976.69  4830.9 1974.04
  4846.8 1971.33  4877.5 1969.89  4911.6 1969.06  4919.5 1967.28  4927.4 1963.01
  4942.5 1959.27    4949 1957.86  4965.3 1956.75  4965.8 1956.25  4988.8 1956.75
  4997.2  1958.8  5023.1  1959.1  5051.2 1962.62    5067 1972.29  5072.8 1973.69
  5080.4 1977.95  5088.6 1983.11  5094.4  1982.7  5110.2 1987.24  5131.8 1988.64
  5161.3 1993.54  5212.5 1996.56  5228.3 1998.39  5300.2 2001.84  5403.2 2004.72
#Mann= 6 ,-1 , 0
    4597      .1       0  4877.5     .07       0  4965.3     .05       0
  4988.8     .07       0  5080.4      .1       0  5300.2     .07       0
Bank Sta=4965.3,4988.8
XS Rating Curve= 0 ,0
Exp/Cntr=0.3,0.1

Type RM Length L Ch R = 1 ,6224    ,521,521,521
BEGIN DESCRIPTION:
Rough Hallow 14.0
END DESCRIPTION:
XS GIS Cut Line= 3
      1847286.76     13981083.43        1846675.       13981325.
      1846275.03       13981325.
#Sta/Elev= 30
  4346.9 1991.46  4443.3 1987.83  4478.4 1984.98  4488.6 1985.26  4586.7 1977.68
  4682.1 1976.66  4743.6 1974.75    4768 1973.47  4819.6 1968.68  4851.8 1966.18
  4886.9 1959.01  4905.9 1958.64    4941 1954.37  4950.9 1954.35  4965.4 1952.04
  4972.4 1952.65  4977.6 1950.44  4978.1 1949.94  5001.9 1950.44  5004.6 1952.61
  5013.1 1953.29  5034.6 1954.28  5044.6  1958.3  5054.6 1976.11  5064.6 1983.01
  5104.6 1989.12  5144.6 1991.87  5214.6  1999.5  5344.6 2006.07  5404.6 2007.39
#Mann= 5 ,-1 , 0
  4346.9      .1       0  4819.6     .07       0  4977.6     .05       0
  5001.9     .07       0  5013.1      .1       0
Bank Sta=4977.6,5001.9
XS Rating Curve= 0 ,0
Exp/Cntr=0.3,0.1

Type RM Length L Ch R = 1 ,5703    ,545,545,545
BEGIN DESCRIPTION:
Rough Hallow 13.0
END DESCRIPTION:
XS GIS Cut Line= 3
      1846924.97       13980825.        1846525.       13980875.
      1846124.98       13980875.
#Sta/Elev= 30
  4596.9 1976.16  4639.7 1974.83  4657.3 1974.88  4720.3 1972.09  4768.2 1969.27
  4838.7  1966.3    4869 1963.12  4888.8 1962.31  4939.5 1958.08  4949.6 1956.59
  4957.1  1953.6  4962.2 1954.54  4969.7  1950.8  4979.8 1947.32  4997.5 1943.76
  4997.8 1941.03  4998.3 1940.53  5021.6 1940.53  5022.1 1941.03    5030 1944.97
    5050 1961.68    5060 1974.72    5070 1986.79    5080 1999.68    5090 2004.89
    5100 2007.24    5110 2007.88    5130 2007.82    5200 2009.47    5400  2016.1
#Mann= 4 ,-1 , 0
  4596.9      .1       0  4888.8     .07       0  4997.8     .05       0
  5022.1     .07       0
Bank Sta=4997.8,5022.1
XS Rating Curve= 0 ,0
Exp/Cntr=0.3,0.1

Type RM Length L Ch R = 1 ,5158    ,486,486,486
BEGIN DESCRIPTION:
Rough Hallow 12.0
END DESCRIPTION:
XS GIS Cut Line= 3
      1847025.03     13980575.02        1846675.     13980381.07
       1846559.2     13980364.14
#Sta/Elev= 30
    4604 1975.03  4626.9  1973.5  4633.8 1973.76  4639.5 1972.49  4649.8  1972.7
  4661.3 1971.37  4715.1 1969.94  4764.3    1964  4827.6 1960.12  4861.3 1957.82
  4867.3 1954.64  4889.8  1947.4  4912.7 1946.57  4921.1 1948.94  4926.9 1949.01
  4958.4 1948.71  4964.6 1947.86  4970.4 1946.91  4980.6 1938.25  4981.1 1937.75
  5004.9 1938.25  5006.7 1940.09  5010.4 1958.56  5034.5 1977.95  5044.6 1989.91
  5054.7 1996.98  5074.9 2005.28  5080.3  2008.2  5105.2 2010.06  5121.2 2009.08
#Mann= 4 ,-1 , 0
    4604      .1       0  4827.6     .07       0  4980.6     .05       0
  5004.9     .07       0
Bank Sta=4980.6,5004.9
XS Rating Curve= 0 ,0
Exp/Cntr=0.3,0.1

Type RM Length L Ch R = 1 ,4672    ,235,235,235
BEGIN DESCRIPTION:
Rough Hallow 11.0
END DESCRIPTION:
XS GIS Cut Line= 3
      1847324.98     13980324.98      1847039.36     13980061.82
      1846875.01       13980025.
#Sta/Elev= 30
  4612.4 1975.35  4640.4 1973.82  4676.2 1968.17  4782.2 1956.09  4853.1 1953.67
  4881.8  1950.7  4888.3 1948.88  4909.8 1947.02  4916.6 1945.26    4924 1944.63
  4938.2 1940.03  4952.3  1940.1  4959.1 1938.84  4980.1 1939.32  4985.5 1938.01
  4985.8 1937.51  4989.5 1938.01  5004.9 1940.92  5015.5 1943.87  5053.1 1943.35
  5066.7 1948.44    5077 1955.33  5087.2 1963.35  5096.5 1976.64  5101.6 1990.43
  5107.7 1996.98    5118 1999.67  5138.5 2002.11  5150.1 2005.02  5169.2 2006.75
#Mann= 4 ,-1 , 0
  4612.4      .1       0  4881.8     .07       0  4985.5     .05       0
  4989.5     .07       0
Bank Sta=4985.5,4989.5
XS Rating Curve= 0 ,0
Exp/Cntr=0.3,0.1

Type RM Length L Ch R = 1 ,4437    ,494,494,494
BEGIN DESCRIPTION:
Rough Hallow 10.0
END DESCRIPTION:
XS GIS Cut Line= 3
      1847483.11     13980269.42      1847243.72     13979945.81
      1847175.01     13979875.01
#Sta/Elev= 30
  4597.5 1984.86  4600.1 1984.86  4627.9  1978.4  4670.7 1975.86    4700 1972.82
  4756.3 1961.19  4764.7 1958.82  4785.5 1955.31  4856.5 1952.06  4871.1 1949.28
  4900.4  1947.2  4935.8 1943.39    4942 1943.98  4952.4 1942.72  4971.3 1940.28
  4985.9 1935.31  4997.4 1930.37  5006.8  1931.2  5018.9 1929.57  5019.2 1929.07
  5022.9 1929.57    5035 1934.79  5042.2  1961.8  5049.2 1966.98  5056.4 1977.27
  5077.5 1989.51    5081 1990.57  5091.6 1993.26  5095.2  1995.2  5098.7  1995.2
#Mann= 5 ,-1 , 0
  4597.5      .1       0  4952.4     .07       0  5018.9     .05       0
  5022.9     .07       0    5081      .1       0
Bank Sta=5018.9,5022.9
XS Rating Curve= 0 ,0
Exp/Cntr=0.3,0.1

Type RM Length L Ch R = 1 ,3943    ,489,489,489
BEGIN DESCRIPTION:
Rough Hallow 9.0
END DESCRIPTION:
XS GIS Cut Line= 3
        1847875.       13979875.      1847661.28     13979681.32
      1847524.98     13979574.98
#Sta/Elev= 30
  4711.4 1986.03  4739.4 1983.29  4775.3 1976.33  4789.5 1972.15  4810.4 1964.01
  4838.8 1954.46  4859.8 1948.24  4867.2 1946.98  4873.9 1944.32  4881.4 1942.71
  4888.1 1939.73  4902.3 1936.27    4924 1936.17  4942.9 1933.36  4943.1 1932.86
  4946.6 1932.86  4946.9 1933.36  4993.9  1934.8    5008 1934.28  5016.2 1935.57
    5037 1944.44  5045.1  1945.9  5072.3 1953.63  5090.9 1957.55  5109.3 1962.54
    5122 1967.65  5136.5 1971.51    5151 1975.04  5169.5 1978.11  5172.7 1978.11
#Mann= 5 ,-1 , 0
  4711.4      .1       0  4859.8     .07       0  4942.9     .05       0
  4946.9     .07       0  5090.9      .1       0
Bank Sta=4942.9,4946.9
XS Rating Curve= 0 ,0
Exp/Cntr=0.3,0.1
