HEC-RAS study South Fork Guadalupe River.prj: South Fork Guadalupe River Base Level Engineering

--- South Fork Guadalupe River.g01 (geometry) --- (continued)

Type RM Length L Ch R = 1 ,56097   ,698,698,698
BEGIN DESCRIPTION:
South Fork Guadalupe River 79.0
END DESCRIPTION:
XS GIS Cut Line= 3
      1838193.21      13910531.6        1838675.       13910525.
      1839364.21     13910289.72
#Sta/Elev= 30
  4518.6 1960.39  4610.4 1963.98  4680.4 1971.05  4730.4 1972.32  4770.4  1970.7
  4790.4 1967.55  4800.5 1964.04  4820.4 1949.34  4830.4 1931.78  4840.4  1921.3
  4860.4 1908.76  4870.4 1904.28  4910.4 1897.61  4980.4 1894.29  4984.5 1891.21
    4986 1890.21  5047.7 1891.21  5049.9  1891.3  5204.1 1893.01    5230 1905.58
  5329.4 1914.17    5402 1925.49  5444.1 1935.96  5449.4 1935.91  5454.8 1938.85
    5512  1955.2  5538.1 1969.87  5574.7 1973.49    5645 1990.26  5728.7 2002.91
#Mann= 6 ,-1 , 0
  4518.6     .07       0  4800.5    .035       0  4984.5    .035       0
  5047.7    .035       0  5049.9     .07       0    5230      .1       0
Bank Sta=4984.5,5047.7
XS Rating Curve= 0 ,0
Exp/Cntr=0.3,0.1

Type RM Length L Ch R = 1 ,55399   ,706,706,706
BEGIN DESCRIPTION:
South Fork Guadalupe River 78.0
END DESCRIPTION:
XS GIS Cut Line= 4
      1837394.57     13910893.77      1838369.71     13911083.94
        1838825.       13911175.      1839324.98       13911275.
#Sta/Elev= 30
  3546.3 2025.28  3658.8 2012.45  3699.6 2005.04  3843.7 1994.52  4209.9 1978.93
  4359.6 1977.36  4545.2 1971.56  4674.1 1952.73  4708.4  1949.9  4718.6 1946.41
  4749.2 1924.13  4769.6 1900.82  4779.8  1896.2  4800.2 1891.35  4871.5 1889.89
  4901.1  1887.3  4902.6  1886.3  4964.3  1887.3  4973.7 1887.43  5006.7 1888.23
  5034.7 1892.38  5062.9 1901.76  5075.5 1905.27  5177.5  1906.7  5228.5 1910.11
  5299.9  1924.7  5422.2 1957.08  5483.4 1968.49  5493.6 1972.02    5514  1972.6
#Mann= 6 ,-1 , 0
  3546.3      .1       0  4674.1    .035       0  4901.1    .033       0
  4964.3    .035       0  4973.7    .033       0  5062.9      .1       0
Bank Sta=4901.1,4964.3
XS Rating Curve= 0 ,0
Exp/Cntr=0.3,0.1

Type RM Length L Ch R = 1 ,54693   ,670,670,670
BEGIN DESCRIPTION:
South Fork Guadalupe River 77.0
END DESCRIPTION:
XS GIS Cut Line= 4
      1837307.71     13912161.14      1838415.97     13911816.81
        1838875.       13911725.      1839374.97       13911725.
#Sta/Elev= 30
  3366.9 1981.81  3856.2 1962.36  4002.8  1958.2  4210.2 1945.69  4264.6 1944.23
  4448.6 1933.66  4505.5 1932.65  4658.3  1923.1  4679.4 1920.74  4740.6 1918.82
  4750.8 1917.22  4771.2 1908.75  4822.2  1892.7    4891 1888.87  4924.1 1887.95
  4944.5 1889.05  4953.1 1887.28  4954.6 1886.28  5017.6 1887.28  5095.5 1888.33
  5125.5 1894.67  5146.6  1902.7  5205.5 1905.58  5225.5 1910.54  5295.5 1937.23
  5325.5 1946.16  5405.5 1961.31  5415.5 1965.07  5435.5  1969.3  5495.5 1974.56
#Mann= 6 ,-1 , 0
  3366.9     .07       0  4658.3    .035       0    4891     .07       0
  4953.1     .05       0  5017.6     .07       0  5146.6      .1       0
Bank Sta=4953.1,5017.6
XS Rating Curve= 0 ,0
Exp/Cntr=0.3,0.1

Type RM Length L Ch R = 1 ,54023   ,674,674,674
BEGIN DESCRIPTION:
South Fork Guadalupe River 76.0
END DESCRIPTION:
XS GIS Cut Line= 3
      1838574.99     13912925.02        1838975.       13912325.
      1839374.98     13912025.02
#Sta/Elev= 30
  4279.6 2008.81  4308.2 2002.95  4338.2 1992.83  4479.1 1932.45  4524.5 1915.35
  4581.6 1903.25  4611.6 1903.49  4794.6 1892.47    4864 1892.23  4915.1 1887.67
  4921.1 1884.86  4936.1 1885.01  4939.9 1882.72  4941.4 1881.72  5004.4 1882.72
    5008 1886.38  5200.7 1886.93  5243.4 1905.12    5258 1916.86  5264.3 1917.71
  5272.6 1924.68  5278.9 1927.14  5287.2 1935.65  5293.4 1936.06  5300.7  1947.6
    5308 1950.14  5364.3 1956.26  5393.4 1961.02    5408 1966.22  5500.7 1971.32
#Mann= 5 ,-1 , 0
  4279.6      .1       0  4479.1    .035       0  4794.6      .1       0
  4939.9     .05       0  5004.4      .1       0
Bank Sta=4939.9,5004.4
XS Rating Curve= 0 ,0
Exp/Cntr=0.3,0.1

Type RM Length L Ch R = 1 ,53349   ,817,817,817
BEGIN DESCRIPTION:
South Fork Guadalupe River 75.0
END DESCRIPTION:
XS GIS Cut Line= 3
      1838624.96     13913025.01        1839225.       13912825.
        1839625.       13912525.
#Sta/Elev= 30
  4375.6 2010.95  4396.7 2008.72  4428.3 2000.83  4454.7 1987.44    4460 1981.44
  4514.9 1952.98  4586.5 1917.37  4618.1 1904.79  4649.7 1897.99  4771.1 1888.22
  4818.4 1888.18  4839.4 1884.14  4909.5 1882.61  4973.2 1882.23  4974.7 1881.23
  5037.8 1882.23  5044.6 1899.04  5050.8 1906.65  5058.1 1911.19  5071.6 1913.66
  5100.8 1918.35  5136.2 1919.05  5150.8 1918.64  5165.4 1912.94  5171.6 1913.24
  5215.4 1926.07  5315.4 1946.89  5350.8  1948.9  5415.4 1958.44  5508.1 1965.06
#Mann= 6 ,-1 , 0
  4375.6      .1       0  4514.9    .035       0  4771.1      .1       0
  4909.5     .07       0  4973.2     .05       0  5037.8      .1       0
Bank Sta=4973.2,5037.8
XS Rating Curve= 0 ,0
Exp/Cntr=0.3,0.1

Type RM Length L Ch R = 1 ,52532   ,594,594,594
BEGIN DESCRIPTION:
South Fork Guadalupe River 74.0
END DESCRIPTION:
XS GIS Cut Line= 3
      1839374.99     13913825.03      1839446.09     13913409.88
      1839975.03     13912824.97
#Sta/Elev= 30
  4569.2 2001.06  4776.9 1983.85  4812.7 1974.06    4837 1964.62  4843.2 1952.13
  4853.3 1937.43  4873.6 1920.39    4897 1893.87  4912.6 1886.51  4957.9 1880.84
  4959.4 1879.84  5022.8 1880.84  5177.1 1883.07  5206.6  1887.5  5219.6 1893.41
  5226.4 1894.12    5340  1893.4  5354.2 1897.22  5368.3 1907.91  5439.3  1923.1
  5502.9 1927.58  5566.4 1923.94  5594.8 1929.54  5616.4 1937.62  5651.6 1945.56
  5694.1 1951.35  5708.3 1950.02  5715.1 1953.75  5722.5 1952.56    5779 1959.69
#Mann= 5 ,-1 , 0
  4569.2     .07       0  4912.6    .035       0  4957.9    .035       0
  5022.8    .035       0  5206.6      .1       0
Bank Sta=4957.9,5022.8
XS Rating Curve= 0 ,0
Exp/Cntr=0.3,0.1

Type RM Length L Ch R = 1 ,51938   ,721,721,721
BEGIN DESCRIPTION:
South Fork Guadalupe River 73.0
END DESCRIPTION:
XS GIS Cut Line= 3
      1839524.96     13913925.03        1839925.       13913625.
      1840025.01     13912924.95
#Sta/Elev= 30
  4495.1 2019.41  4631.6 2003.18  4723.3    1988  4790.7 1972.65  4852.4 1960.03
  4881.6 1951.41  4895.1 1935.28  4902.4 1932.33  4908.7 1898.29    4917 1892.89
  4923.3 1882.47  4931.6 1881.89  4934.6 1879.54  4936.1 1878.54  4999.5 1879.54
  5100.4 1880.51  5197.2 1881.08  5207.3 1882.39  5223.3 1889.98  5237.6 1896.29
  5247.7 1896.49  5267.9 1889.53    5278 1888.64  5319.4 1890.46  5368.9 1891.25
  5409.3 1897.67  5459.8 1901.59  5538.1 1923.85  5621.4 1943.49  5702.3 1953.45
#Mann= 8 ,-1 , 0
  4495.1     .07       0  4790.7      .1       0  4934.6     .05       0
  4999.5      .1       0  5100.4    .033       0  5223.3      .1       0
  5319.4    .035       0  5538.1      .1       0
Bank Sta=4934.6,4999.5
XS Rating Curve= 0 ,0
Exp/Cntr=0.3,0.1

Type RM Length L Ch R = 1 ,51217   ,715,715,715
BEGIN DESCRIPTION:
South Fork Guadalupe River 72.0
END DESCRIPTION:
XS GIS Cut Line= 3
      1840774.99     13913824.98        1840475.       13913425.
        1840475.     13912924.98
#Sta/Elev= 30
  4503.9 2063.23    4582 2050.15    4631 2035.42  4646.6 2030.42  4661.2 2020.08
  4696.6 2008.08  4711.2  1996.2    4732 1987.84  4740.3 1980.04  4746.6 1979.55
  4761.2 1967.31  4767.4 1966.74    4782 1955.29  4790.3 1931.82  4803.9 1922.26
  4811.2 1910.27  4817.4 1906.03  4825.8 1892.93    4832 1891.07  4840.3 1874.55
  4968.3 1873.21  4969.8 1872.21  5033.3 1873.21  5033.9 1876.16  5093.9 1882.98
    5125 1891.33  5269.2 1897.76  5323.9  1901.6  5393.9 1926.41  5503.9 1949.93
#Mann= 6 ,-1 , 0
  4503.9      .1       0    4631     .07       0  4968.3    .033       0
  5033.3     .07       0    5125      .1       0  5269.2    .035       0
Bank Sta=4968.3,5033.3
XS Rating Curve= 0 ,0
Exp/Cntr=0.3,0.1

Type RM Length L Ch R = 1 ,50502   ,654,654,654
BEGIN DESCRIPTION:
South Fork Guadalupe River 71.0
END DESCRIPTION:
XS GIS Cut Line= 3
        1841125.     13913825.04        1841125.       13913325.
      1841025.01     13912825.05
#Sta/Elev= 30
  4495.1 2073.42  4515.1  2064.1  4555.1 2050.21  4605.1 2027.93  4625.1 2021.37
  4765.1 1951.99  4855.1 1905.25  4875.1 1882.92  4895.1 1876.51  4925.1 1870.59
  4973.5 1868.85  4992.6 1870.03  4993.2  1868.7  4994.7  1867.7  5058.2  1868.7
  5086.9 1868.88  5117.5 1873.81  5127.7 1875.98  5158.3 1889.01  5168.5 1890.33
  5188.9 1892.13  5252.3  1892.1  5290.9 1894.73  5311.3 1903.05  5331.7  1916.6
  5352.1 1925.92  5382.7 1938.57  5403.1 1944.98  5433.7 1950.22    5505 1955.48
#Mann= 5 ,-1 , 0
  4495.1      .1       0  4973.5     .07       0  4993.2     .05       0
  5058.2     .07       0  5252.3    .035       0
Bank Sta=4993.2,5058.2
XS Rating Curve= 0 ,0
Exp/Cntr=0.3,0.1

Type RM Length L Ch R = 1 ,49848   ,709,709,709
BEGIN DESCRIPTION:
South Fork Guadalupe River 70.0
END DESCRIPTION:
XS GIS Cut Line= 3
        1841625.     13913775.01        1841625.       13913175.
      1841246.79     13912862.22
#Sta/Elev= 30
  4404.3 2049.94  4444.3 2038.32  4554.3 1996.11  4664.3 1949.96  4734.3  1917.2
  4794.3 1896.38  4814.3 1872.45  4820.2 1871.26  4935.9 1868.71  4961.8 1868.53
  4963.3 1867.53  5026.8 1868.53  5032.3  1874.1  5040.1 1874.51  5046.6 1878.07
  5101.9 1887.79  5255.7 1891.73    5289 1891.44  5316.3 1897.67  5324.1 1896.33
  5330.6 1891.72  5367.1 1893.06  5387.9 1903.84  5394.4 1909.76  5402.3 1911.99
  5408.8 1918.59  5416.6 1920.59  5423.1  1926.5  5437.4 1932.68  5495.1 1946.27
#Mann= 7 ,-1 , 0
  4404.3      .1       0  4820.2     .07       0  4935.9    .033       0
  4961.8    .033       0  5026.8    .033       0  5101.9      .1       0
  5255.7    .035       0
Bank Sta=4961.8,5026.8
XS Rating Curve= 0 ,0
Exp/Cntr=0.3,0.1

Type RM Length L Ch R = 1 ,49139   ,713,713,713
BEGIN DESCRIPTION:
South Fork Guadalupe River 69.0
END DESCRIPTION:
XS GIS Cut Line= 3
        1842125.     13913824.99        1842225.       13913325.
        1842225.     13912824.99
#Sta/Elev= 30
  4490.2 2025.83  4561.6 2024.71    4633 2017.65    4684 2007.68  4724.7 1994.71
  4755.3 1982.28  4806.3 1958.85  4867.5 1921.95  4898.1 1906.93  4944.2 1876.08
  4959.3  1870.9  4979.7 1867.76  5043.3 1868.14  5127.5 1867.53    5129 1866.53
  5191.2 1866.53  5192.7 1867.53  5200.1 1876.09  5226.3 1880.19  5280.1 1883.43
  5370.1 1884.86  5373.2 1886.24  5390.1 1893.97  5400.1 1902.68  5410.1 1914.33
  5420.1 1922.11  5430.1 1927.64  5460.1 1938.48  5480.1 1940.83  5500.1 1941.12
#Mann= 7 ,-1 , 0
  4490.2      .1       0  4944.2    .033       0  5043.3     .07       0
  5127.5    .033       0  5192.7     .07       0  5226.3      .1       0
  5373.2    .035       0
Bank Sta=5127.5,5192.7
XS Rating Curve= 0 ,0
Exp/Cntr=0.3,0.1

Type RM Length L Ch R = 1 ,48426   ,716,716,716
BEGIN DESCRIPTION:
South Fork Guadalupe River 68.0
END DESCRIPTION:
XS GIS Cut Line= 3
      1842525.01     13913774.99        1842825.       13913275.
        1842825.     13912774.98
#Sta/Elev= 30
  4412.5 1991.08  4478.6 1991.95  4595.2 1985.97  4659.3 1973.19  4696.3 1963.63
  4711.8 1956.81  4717.6 1957.38  4748.7 1940.91  4754.6 1940.68    4807 1917.96
  4812.9 1917.74  4828.4 1907.91  4834.3 1907.95  4886.7 1886.17  4913.9 1877.25
  4923.7 1871.82    4928 1865.26  4929.5 1864.26  4993.2 1865.26  5029.7 1866.18
  5185.6 1865.34  5245.6 1878.66  5315.6  1876.9  5323.9 1878.39  5335.6 1882.97
  5345.6 1898.92  5355.6 1908.16  5375.6 1916.13  5425.6  1927.5  5495.6 1930.61
#Mann= 5 ,-1 , 0
  4412.5      .1       0    4928     .05       0  4993.2      .1       0
  5029.7     .07       0  5323.9    .035       0
Bank Sta=4928,4993.2
XS Rating Curve= 0 ,0
Exp/Cntr=0.3,0.1

Type RM Length L Ch R = 1 ,47710   ,664,664,664
BEGIN DESCRIPTION:
South Fork Guadalupe River 67.0
END DESCRIPTION:
XS GIS Cut Line= 3
      1843525.01     13913425.03        1843325.       13912925.
        1843325.     13912424.95
#Sta/Elev= 30
  4460.8 1979.18  4493.1 1971.54  4514.7 1964.75  4529.5 1944.63  4536.2 1930.75
  4553.7 1914.62  4568.5 1907.96  4590.1 1895.49  4600.9  1890.4  4631.8 1883.24
  4729.9 1877.72  4744.9 1875.81  4774.5 1869.03  4783.9 1865.58  4793.4 1864.02
  5006.7 1863.48  5008.2 1862.48  5070.5 1862.48    5072 1863.48  5079.4 1871.45
  5119.4 1871.86  5127.9 1873.55  5139.4 1878.02  5159.4 1889.39  5169.4 1907.76
  5179.4 1915.78  5199.4 1922.42  5229.4 1929.58  5337.8 1937.19  5499.4 1945.28
#Mann= 6 ,-1 , 0
  4460.8      .1       0  4729.9     .07       0  5006.7     .05       0
    5072     .07       0  5127.9    .035       0  5337.8      .1       0
Bank Sta=5006.7,5072
XS Rating Curve= 0 ,0
Exp/Cntr=0.3,0.1

Type RM Length L Ch R = 1 ,47046   ,704,704,704
BEGIN DESCRIPTION:
South Fork Guadalupe River 66.0
END DESCRIPTION:
XS GIS Cut Line= 3
      1844125.01     13913225.01        1843925.       13912725.
      1843525.03     13912425.02
#Sta/Elev= 30
  4460.9 1961.24  4505.3 1954.33  4528.2  1946.2  4547.1 1926.66  4553.8 1916.72
  4559.2 1911.75    4613 1880.87  4631.9    1879  4708.6 1879.79  4798.8 1873.49
  4823.7  1866.2  4852.7 1859.94  4945.2 1859.02  4946.7 1858.02  5010.5 1859.02
  5106.7 1860.23  5127.6 1863.08  5171.3 1864.12  5177.6 1869.15  5185.9 1871.37
  5192.1 1882.68    5196 1883.18  5206.7 1884.81    5213 1898.19  5235.9 1904.94
  5242.1 1908.93  5306.7 1922.23  5356.7 1929.51  5394.8 1931.46  5499.4 1938.84
#Mann= 6 ,-1 , 0
  4460.9      .1       0  4823.7     .07       0  4945.2     .05       0
  5010.5     .07       0    5196    .035       0  5394.8      .1       0
Bank Sta=4945.2,5010.5
XS Rating Curve= 0 ,0
Exp/Cntr=0.3,0.1

Type RM Length L Ch R = 1 ,46342   ,682,682,682
BEGIN DESCRIPTION:
South Fork Guadalupe River 65.0
END DESCRIPTION:
XS GIS Cut Line= 3
      1844624.99     13912924.98        1844425.       13912425.
        1844125.       13912025.
#Sta/Elev= 30
  4465.3 1964.46  4480.1 1962.85  4509.7 1953.83  4519.1 1942.65  4533.9 1929.63
  4540.7 1902.31  4551.4 1898.34    4573 1882.36  4594.5 1873.17    4612 1872.91
  4648.4 1879.48  4702.2 1882.01  4725.1 1880.78  4773.6 1863.85  4820.7 1859.29
  4884.1 1859.64  4956.3  1858.8  4957.8  1857.8  5021.7  1858.8  5025.7 1862.43
  5061.1 1862.46  5076.7 1865.34    5091 1867.16  5117.3 1874.16  5146.5 1891.28
  5161.1 1901.95  5190.3  1913.4  5305.4 1929.72  5340.3 1934.92  5503.8 1944.59
#Mann= 7 ,-1 , 0
  4465.3      .1       0  4884.1    .033       0  4956.3    .033       0
  5021.7    .033       0  5076.7     .07       0    5091    .035       0
  5305.4      .1       0
Bank Sta=4956.3,5021.7
XS Rating Curve= 0 ,0
Exp/Cntr=0.3,0.1

Type RM Length L Ch R = 1 ,45660   ,704,704,704
BEGIN DESCRIPTION:
South Fork Guadalupe River 64.0
END DESCRIPTION:
XS GIS Cut Line= 3
        1845025.     13912875.01        1845025.       13912375.
      1844625.01     13911875.02
#Sta/Elev= 30
  4495.6 1969.81  4505.6 1970.12  4628.4 1962.61  4735.6 1955.26  4754.6 1951.07
  4805.6 1932.25  4855.6 1911.37  4875.6 1899.78  4885.6 1891.08  4895.6  1870.9
  4905.6 1868.67  4965.6  1860.9  4998.8 1861.21  5019.7    1859  5021.2    1858
  5083.6    1858  5085.1    1859  5223.7  1859.8  5234.2 1860.76  5294.2 1867.75
  5308.6 1870.37  5329.4 1877.22  5363.6 1878.63  5372.6 1877.97  5430.2 1882.39
  5457.4 1893.44  5500.7 1918.16  5524.7 1924.91  5585.5 1936.35  5635.9 1939.46
#Mann= 8 ,-1 , 0
  4495.6      .1       0  4628.4     .07       0  4754.6      .1       0
  5019.7     .05       0  5085.1      .1       0  5234.2     .07       0
  5363.6    .035       0  5524.7      .1       0
Bank Sta=5019.7,5085.1
XS Rating Curve= 0 ,0
Exp/Cntr=0.3,0.1

Type RM Length L Ch R = 1 ,44956   ,584,584,584
BEGIN DESCRIPTION:
South Fork Guadalupe River 63.0
END DESCRIPTION:
XS GIS Cut Line= 3
        1845625.     13912574.99        1845625.       13912075.
        1844625.       13911075.
#Sta/Elev= 30
  4495.2  1947.3  4614.8 1940.19  4785.2 1929.14  4895.2 1911.64  4935.2 1895.39
  4945.2 1888.25  4965.2 1866.34  4975.2 1860.43  4990.8 1858.79  4992.3 1857.79
  5056.2 1858.79  5225.2 1860.34  5235.6 1860.21  5263.9  1870.2  5292.2 1875.66
  5368.9 1880.03  5554.6 1879.41  5673.3 1880.84  5688.2 1882.48  5716.4 1893.21
  5787.2 1936.29  5801.3 1941.19  5886.1 1955.67  5968.8 1959.83    6070 1973.13
  6098.3  1979.9  6154.7 1984.96  6183.1 1992.91  6239.7 2002.68  6409.4 2026.25
#Mann= 10 ,-1 , 0
  4495.2     .07       0  4614.8      .1       0  4990.8     .05       0
  5056.2      .1       0  5225.2      .1       0  5368.9    .035       0
  5554.6     .07       0  5673.3      .1       0  5968.8     .07       0
  6154.7      .1       0
Bank Sta=4990.8,5056.2
XS Rating Curve= 0 ,0
Exp/Cntr=0.3,0.1

Type RM Length L Ch R = 1 ,44372   ,60,60,60
BEGIN DESCRIPTION:
South Fork Guadalupe River 62.0
END DESCRIPTION:
XS GIS Cut Line= 3
      1846224.99     13912124.98      1846084.64     13911753.18
      1845525.01     13911125.02
#Sta/Elev= 30
  4612.5 1939.34  4644.4 1938.69  4751.4 1936.51  4847.6 1930.24  4901.1 1917.88
  4924.3 1907.91  4943.8 1895.67  4963.1 1887.01    4966 1859.02  4967.5 1858.02
  5031.4 1859.02  5219.1 1860.96  5248.8 1870.65  5277.2 1875.39  5357.7 1876.21
  5462.1 1876.78    5605 1875.74  5666.9 1877.52  5695.3 1892.16  5702.8 1899.04
  5709.5 1900.82    5717 1908.88  5730.7 1919.08  5737.9 1929.88  5752.1  1938.7
  5766.4 1953.67  5801.5 1957.39    5809 1961.82  5850.1 1963.82  5851.2 1963.82
#Mann= 10 ,-1 , 0
  4612.5      .1       0  4644.4     .07       0  4924.3      .1       0
    4966     .05       0  5031.4      .1       0  5219.1     .07       0
  5357.7    .063       0  5462.1    .035       0    5605      .1       0
  5850.1     .07       0
Bank Sta=4966,5031.4
XS Rating Curve= 0 ,0
Exp/Cntr=0.3,0.1

Type RM Length L Ch R = 1 ,44312   ,782,782,782
BEGIN DESCRIPTION:
South Fork Guadalupe River 81.1
END DESCRIPTION:
XS GIS Cut Line= 4
      1846282.08     13912146.84      1846138.87     13911739.33
      1845994.34     13911504.96      1845638.77     13911153.28
#Sta/Elev= 30
  4539.6 1939.86  4630.6  1937.8  4721.6 1937.36  4788.9 1933.17  4838.3 1928.92
  4869.6 1921.19  4901.9 1911.26  4912.8 1903.54  4933.2 1894.23  4954.9 1879.35
  4969.5  1859.7    4974 1859.09  4975.5 1858.09  5039.4 1859.09  5176.9  1859.8
  5201.9 1860.62  5232.7 1869.78  5243.9 1875.51  5340.2 1876.06  5492.4 1876.81
  5621.2 1874.93  5649.5  1880.5  5671.7 1893.67  5691.9 1906.23  5698.9 1916.69
    5706 1919.35  5727.2 1941.45  5734.3  1944.2  5741.4 1953.46    5747 1954.29
#Mann= 9 ,-1 , 0
  4539.6      .1       0  4630.6     .07       0  4869.6      .1       0
    4974     .05       0  5039.4      .1       0  5176.9     .07       0
  5340.2    .063       0  5492.4    .035       0  5671.7      .1       0
Bank Sta=4974,5039.4
XS Rating Curve= 0 ,0
Exp/Cntr=0.3,0.1

Type RM Length L Ch R = 1 ,43530   ,718,718,718
BEGIN DESCRIPTION:
South Fork Guadalupe River 61.0
END DESCRIPTION:
XS GIS Cut Line= 3
      1846474.99     13911775.03        1846575.       13911275.
      1846114.97     13910905.47
#Sta/Elev= 30
  4495.2 1928.97    4587 1926.48    4619 1923.78  4648.2 1920.88  4678.8 1914.53
  4719.6 1895.03    4740 1889.06  4770.6 1855.68  4801.2 1852.32  4923.5 1853.64
    4952 1851.49  4953.5 1850.49  5017.4 1851.49  5029.7 1852.62  5076.3 1858.11
  5082.7 1857.22  5204.3 1866.68  5239.5  1871.9  5410.7  1872.4  5439.5  1875.5
    5446 1879.59  5453.9 1881.67  5460.4 1887.44  5474.7 1892.95  5481.2 1903.23
  5489.1 1907.74  5495.6 1914.98  5526.1  1923.7  5559.6 1929.23  5595.2 1929.86
#Mann= 6 ,-1 , 0
  4495.2     .07       0    4619      .1       0    4952     .05       0
  5017.4      .1       0  5029.7    .035       0  5526.1     .07       0
Bank Sta=4952,5017.4
XS Rating Curve= 0 ,0
Exp/Cntr=0.3,0.1

Type RM Length L Ch R = 1 ,42812   ,714,714,714
BEGIN DESCRIPTION:
South Fork Guadalupe River 60.0
END DESCRIPTION:
XS GIS Cut Line= 3
      1846824.98     13911575.02        1847225.       13911275.
        1847225.     13910675.03
#Sta/Elev= 30
  4492.2  1919.3  4528.7 1913.16  4549.5 1906.71  4584.9 1888.51  4620.4 1877.05
  4677.5 1872.93  4699.5 1872.19  4705.8  1867.7  4714.1 1868.81  4720.4 1865.11
  4728.7 1868.49  4734.9  1864.5  4749.5 1868.22  4755.8 1863.34  4764.1 1862.69
  4814.1 1865.64  4894.4 1862.69  4920.4 1855.17  4978.5 1851.64    4980 1850.64
  5045.9 1851.64  5081.5 1852.01  5172.2 1852.03  5252.2 1856.58  5262.2 1874.34
    5273  1882.9  5322.2 1905.04  5472.2 1947.92  5567.3 1967.43  5592.2 1971.09
#Mann= 8 ,-1 , 0
  4492.2      .1       0  4677.5    .035       0  4894.4      .1       0
  4978.5     .05       0  5045.9      .1       0  5081.5    .033       0
    5273      .1       0  5567.3     .07       0
Bank Sta=4978.5,5045.9
XS Rating Curve= 0 ,0
Exp/Cntr=0.3,0.1

Type RM Length L Ch R = 1 ,42098   ,80,80,80
BEGIN DESCRIPTION:
South Fork Guadalupe River 59.0
END DESCRIPTION:
XS GIS Cut Line= 3
      1847075.04     13912024.98        1847675.       13911725.
      1847975.01     13911324.98
#Sta/Elev= 30
    4329 1910.87  4330.3 1910.87  4387.7 1909.27    4459 1894.79  4519.7 1879.92
  4544.2 1872.71  4631.7  1871.1  4805.6 1871.06    4888  1867.6  4910.3  1863.9
  4929.7 1851.92  4931.2 1850.92  4997.2 1851.92  5207.1  1854.4  5213.3 1867.47
  5221.7  1864.1  5227.9 1940.91  5236.2 1938.15  5242.5 1954.22  5257.1 1960.52
  5263.3 1969.06  5271.7 1971.65  5277.9 1978.13  5286.2  1980.4  5292.5 1989.24
  5307.1 1995.76  5313.3 2002.72  5354.5 2010.47  5470.6 2017.08  5499.8  2017.8
#Mann= 10 ,-1 , 0
    4329     .07       0  4330.3      .1       0    4459     .07       0
  4519.7      .1       0  4631.7    .035       0  4805.6     .07       0
  4929.7     .05       0  4997.2     .07       0  5354.5      .1       0
  5470.6     .07       0
Bank Sta=4929.7,4997.2
XS Rating Curve= 0 ,0
Exp/Cntr=0.3,0.1

Type RM Length L Ch R = 1 ,42018   ,527,527,527
BEGIN DESCRIPTION:
South Fork Guadalupe River 59.1
END DESCRIPTION:
XS GIS Cut Line= 4
      1847142.55     13912055.58      1847619.51     13911811.21
      1847899.89     13911746.97      1848399.07      13911443.6
#Sta/Elev= 30
  4357.2 1907.76  4382.4 1906.31  4449.8 1892.29  4472.3 1887.11  4500.7 1875.22
  4522.9 1871.57  4583.5 1870.64  4792.1 1870.12  4865.6 1868.48  4893.1 1860.87
  4895.8 1852.25  4897.3 1851.25  4963.3 1852.25  5000.7  1858.7    5078 1863.59
  5120.9 1869.54    5126 1866.22  5134.7 1867.53  5163.8 1911.51  5175.7 1921.57
  5180.8 1921.57  5193.4 1939.36  5199.2 1941.71  5208.9 1951.59  5214.7 1952.93
  5218.5 1958.12  5245.2 1986.27  5272.9 1991.31    5674 1992.74  5764.9 1995.48
#Mann= 7 ,-1 , 0
  4357.2      .1       0  4583.5    .035       0  4792.1     .07       0
  4895.8     .05       0  4963.3     .07       0  5000.7    .033       0
  5218.5      .1       0
Bank Sta=4895.8,4963.3
XS Rating Curve= 0 ,0
Exp/Cntr=0.3,0.1

Type RM Length L Ch R = 1 ,41491   ,791,791,791
BEGIN DESCRIPTION:
South Fork Guadalupe River 58.0
END DESCRIPTION:
XS GIS Cut Line= 3
      1847223.36     13912348.91      1847939.24     13912204.82
      1848375.04     13912375.02
#Sta/Elev= 30
  4283.6 1905.34  4336.3 1894.95  4387.5  1878.1  4417.9 1870.06  4492.5 1868.43
  4697.8 1867.83  4736.7 1867.14  4798.7 1848.99  4815.7 1842.82  4924.4 1842.09
    4952 1841.79  4953.5 1840.79  5019.5 1841.79  5041.5 1910.42  5051.2 1918.71
  5056.6 1917.81  5073.7 1937.14  5081.1 1951.68  5086.4 1949.99  5105.2 1959.71
  5234.7 1957.88  5303.7 1950.98  5328.2 1938.04  5333.6 1940.11  5363.6 1921.05
  5382.6  1930.8  5387.9 1924.27  5412.4 1938.02  5416.8  1935.2  5481.7 1951.59
#Mann= 10 ,-1 , 0
  4283.6      .1       0  4387.5     .07       0  4492.5    .035       0
  4697.8      .1       0  4798.7    .033       0  4924.4     .07       0
    4952     .05       0  5019.5     .07       0  5105.2     .07       0
  5416.8      .1       0
Bank Sta=4952,5019.5
XS Rating Curve= 0 ,0
Exp/Cntr=0.3,0.1

Type RM Length L Ch R = 1 ,40700   ,698,698,698
BEGIN DESCRIPTION:
South Fork Guadalupe River 57.0
END DESCRIPTION:
XS GIS Cut Line= 3
      1847075.02       13912825.        1847975.       13912825.
      1848475.02       13912925.
#Sta/Elev= 30
  4099.1 1939.02  4249.1 1909.15  4299.1  1894.9  4313.5 1888.59  4339.1 1879.64
  4389.1  1870.6  4538.5 1864.82  4709.1  1861.4  4749.1 1859.24  4764.6 1856.14
  4819.1 1849.95  4829.1 1843.82  4859.1 1836.66  4954.6 1835.63  4955.3 1835.62
  4956.8 1834.62  5022.8 1835.62  5029.7 1917.83  5039.9 1921.72  5070.5 1925.73
  5121.5 1924.67  5172.4 1915.93  5223.4 1902.93  5264.2 1876.13  5274.4 1873.81
  5325.4  1904.6  5376.4  1924.9  5447.8 1947.14  5486.2  1950.6    5509  1951.5
#Mann= 8 ,-1 , 0
  4099.1      .1       0  4313.5     .07       0  4538.5    .035       0
  4764.6      .1       0  4954.6    .033       0  4955.3     .05       0
  5022.8    .033       0  5486.2     .07       0
Bank Sta=4955.3,5022.8
XS Rating Curve= 0 ,0
Exp/Cntr=0.3,0.1

Type RM Length L Ch R = 1 ,40002   ,718,718,718
BEGIN DESCRIPTION:
South Fork Guadalupe River 56.0
END DESCRIPTION:
XS GIS Cut Line= 3
      1847074.98       13913325.        1847875.       13913325.
      1848374.98       13913325.
#Sta/Elev= 30
    4200  1940.1  4259.8 1934.17    4350 1915.32    4400  1897.9    4450 1877.61
    4480 1868.06  4567.3 1864.76  4621.6 1863.38  4720.2 1862.67    4790 1859.68
    4810 1855.73    4840  1854.7    4860 1850.66  4889.8 1847.83    4920 1846.45
  4926.3 1835.56  4927.8 1834.56  4993.8 1835.56    5055 1836.34  5076.6 1837.59
    5080 1837.93    5090 1883.12    5100 1907.52    5110 1913.07    5140 1917.45
    5190 1917.27  5244.5 1920.15    5350 1933.35    5430  1939.1    5500 1949.66
#Mann= 11 ,-1 , 0
    4200     .07       0  4259.8      .1       0  4567.3     .07       0
  4621.6      .1       0  4720.2    .035       0  4889.8      .1       0
  4926.3     .05       0  4993.8      .1       0    5055    .033       0
  5076.6      .1       0  5244.5     .07       0
Bank Sta=4926.3,4993.8
XS Rating Curve= 0 ,0
Exp/Cntr=0.3,0.1

Type RM Length L Ch R = 1 ,39284   ,674,674,674
BEGIN DESCRIPTION:
South Fork Guadalupe River 55.0
END DESCRIPTION:
XS GIS Cut Line= 3
      1847125.01       13913625.        1847725.       13913925.
      1848224.99       13913825.
#Sta/Elev= 30
    4321 1926.71  4432.8 1912.44  4491.5 1895.33  4508.3 1878.69  4530.6 1870.28
    4553 1864.29  4589.1 1862.75  4714.3 1861.45  4737.5 1860.02  4754.2 1851.34
  4759.8  1853.5  4768.2 1845.63  4776.6 1843.26  4814.5 1843.69  4822.7 1845.61
  4888.4  1849.2  4924.7 1847.43  4961.1 1841.51  4968.3 1835.41  4969.8 1834.41
  5035.8 1835.41  5036.1 1835.43  5137.3 1838.35  5165.2 1850.61  5226.4 1862.42
    5257 1876.97  5287.6 1879.55  5307.9  1891.6  5328.3  1898.9  5501.7 1923.09
#Mann= 9 ,-1 , 0
    4321      .1       0  4589.1     .07       0  4714.3      .1       0
  4814.5     .07       0  4822.7    .035       0  4968.3    .035       0
  5035.8    .035       0  5036.1    .033       0  5137.3      .1       0
Bank Sta=4968.3,5035.8
XS Rating Curve= 0 ,0
Exp/Cntr=0.3,0.1

Type RM Length L Ch R = 1 ,38610   ,715,715,715
BEGIN DESCRIPTION:
South Fork Guadalupe River 54.0
END DESCRIPTION:
XS GIS Cut Line= 3
      1847025.01       13914575.        1847525.       13914475.
      1848425.02     13914074.99
#Sta/Elev= 30
  4483.6 1936.03    4576 1934.63    4657 1929.56  4697.7 1924.42  4728.3 1918.14
  4769.1 1900.15  4809.9 1874.78  4830.3 1864.96  4881.3 1854.49  4901.7 1846.35
  4922.1 1833.47  4939.1 1831.98  4940.6 1830.98    5007 1831.98  5075.6 1835.37
  5168.6    1835  5212.4 1838.62  5234.2 1838.31  5251.3 1845.62  5256.8 1845.26
  5277.2 1851.84  5310.8 1854.51  5562.5 1860.46  5598.8 1869.93    5622 1880.24
  5645.3 1896.05  5650.8 1898.19  5743.8 1913.16  5913.4 1932.83  5978.4  1939.2
#Mann= 7 ,-1 , 0
  4483.6     .07       0    4576      .1       0  4939.1     .05       0
    5007      .1       0  5075.6    .035       0  5277.2      .1       0
  5913.4     .07       0
Bank Sta=4939.1,5007
XS Rating Curve= 0 ,0
Exp/Cntr=0.3,0.1

Type RM Length L Ch R = 1 ,37895   ,688,688,688
BEGIN DESCRIPTION:
South Fork Guadalupe River 53.0
END DESCRIPTION:
XS GIS Cut Line= 3
      1847325.02     13915474.97        1847625.       13915075.
      1848524.99     13914275.01
#Sta/Elev= 30
  4504.8 1959.72  4626.6 1952.26  4712.1 1938.26  4747.5  1935.3  4782.9 1927.19
  4791.2 1920.42  4797.5 1908.72  4804.8 1876.95  4812.1  1875.3  4841.2 1859.22
  4847.5 1850.95  4868.3 1838.54  4882.9 1833.93  4920.8 1832.11  4922.3 1831.11
  4988.7 1832.11  5181.6 1847.29  5189.1 1850.92  5195.8 1849.81  5203.4 1854.73
  5217.6 1856.61  5414.8 1859.37  5639.9 1859.92  5805.4 1860.68  5826.3 1863.14
  5849.1    1871  5911.6 1897.37  6088.5 1922.32  6173.4 1932.63  6208.9 1934.27
#Mann= 6 ,-1 , 0
  4504.8     .07       0  4920.8     .05       0  4988.7     .07       0
  5414.8    .035       0  5639.9     .07       0  5849.1      .1       0
Bank Sta=4920.8,4988.7
XS Rating Curve= 0 ,0
Exp/Cntr=0.3,0.1

Type RM Length L Ch R = 1 ,37207   ,715,715,715
BEGIN DESCRIPTION:
South Fork Guadalupe River 52.0
END DESCRIPTION:
XS GIS Cut Line= 3
      1847475.04     13915674.99        1847975.       13915575.
      1848674.99     13914875.01
#Sta/Elev= 30
  4495.5 1968.77  4556.7 1968.18  4603.7 1962.23  4719.8 1949.25  4740.2 1943.18
  4821.8 1927.19    4832 1908.04  4842.2 1855.35  4852.4 1851.02  4872.8 1846.93
    4883 1838.02  4893.2 1833.05    5028  1831.7  5029.5  1830.7  5095.9  1831.7
  5104.4 1839.67  5132.6  1856.5  5146.8 1859.01  5179.1 1859.04  5619.6 1858.41
    5769 1858.57  5811.5 1855.23  5841.3 1849.86  5853.9 1850.09  5889.2 1865.63
  5896.3 1872.21  5910.5 1881.08  5924.6 1895.23    5960 1905.92  5995.3 1912.66
#Mann= 7 ,-1 , 0
  4495.5     .07       0  4603.7      .1       0    5028     .05       0
  5095.9      .1       0  5179.1      .1       0  5619.6    .035       0
  5841.3      .1       0
Bank Sta=5028,5095.9
XS Rating Curve= 0 ,0
Exp/Cntr=0.3,0.1

Type RM Length L Ch R = 1 ,36492   ,702,702,702
BEGIN DESCRIPTION:
South Fork Guadalupe River 51.0
END DESCRIPTION:
XS GIS Cut Line= 3
        1848325.     13916475.01        1848425.       13915975.
      1849124.98     13915175.02
#Sta/Elev= 30
  4490.1 1946.87  4541.1  1938.1  4673.7 1924.03    4796 1903.94  4887.8 1895.08
    4898 1885.52  4908.2 1854.01  4918.4 1841.21  4925.2 1828.18  4926.7 1827.18
  4993.3 1828.18  5086.8 1830.37  5113.2 1830.36  5254.8 1841.01  5283.3 1847.79
  5290.9 1852.62  5318.9 1856.46  5538.6  1857.9  5691.4 1855.55  5751.2 1853.13
  5793.9 1844.07  5822.4 1844.87  5843.3 1852.09    5886 1880.37  5914.5 1894.63
  5921.1 1895.32  5960.3    1909  5978.1 1914.25  6013.2 1919.17    6063 1920.54
#Mann= 7 ,-1 , 0
  4490.1      .1       0  4925.2     .05       0  4993.3      .1       0
  5086.8    .033       0  5113.2      .1       0  5691.4    .035       0
  5960.3      .1       0
Bank Sta=4925.2,4993.3
XS Rating Curve= 0 ,0
Exp/Cntr=0.3,0.1

Type RM Length L Ch R = 1 ,35790   ,698,698,698
BEGIN DESCRIPTION:
South Fork Guadalupe River 50.0
END DESCRIPTION:
XS GIS Cut Line= 3
        1849325.       13916475.        1849025.       13916075.
        1849325.       13915275.
#Sta/Elev= 30
    4500 2002.15  4561.1 2000.95  4713.5 1990.92  4742.7 1986.26  4842.7 1957.43
  4857.3 1943.34  4892.7 1930.27  4907.3 1908.33  4913.5 1905.73  4921.9 1859.55
  4928.1 1869.56  4936.5  1839.2  4971.9 1829.61  5037.1 1829.83    5127 1828.88
  5128.5 1827.88  5195.1 1828.88  5202.9  1835.4  5224.8 1838.11  5309.7 1839.74
  5341.8 1851.81  5363.1 1854.18  5467.3  1854.1  5556.9 1846.29  5613.2 1845.53
  5643.5 1851.43  5698.7 1875.28  5715.6 1890.06    5780 1911.12  5854.4 1922.27
#Mann= 8 ,-1 , 0
    4500     .07       0  4561.1      .1       0  5037.1    .033       0
    5127     .05       0  5195.1    .033       0  5224.8      .1       0
  5556.9    .035       0    5780      .1       0
Bank Sta=5127,5195.1
XS Rating Curve= 0 ,0
Exp/Cntr=0.3,0.1

Type RM Length L Ch R = 1 ,35092   ,684,684,684
BEGIN DESCRIPTION:
South Fork Guadalupe River 49.0
END DESCRIPTION:
XS GIS Cut Line= 3
        1849525.     13916475.02        1849625.       13915975.
        1849525.     13915275.03
#Sta/Elev= 30
  4485.2 1990.19  4558.1 1988.12  4638.2 1980.95  4699.4 1969.54    4730 1959.44
  4750.4 1945.73  4821.4  1913.9  4872.7 1886.16  4882.9  1876.8  4893.1 1853.99
  4904.3 1846.01  4913.5 1839.23  4933.9 1831.54  4981.1 1828.94  5041.9 1828.56
  5043.4 1827.56    5110 1828.56  5166.9 1832.12  5197.2 1843.52  5211.6 1844.37
  5227.5 1841.78  5267.9 1846.31  5301.1 1845.34  5348.7 1845.62    5480 1854.78
  5510.3 1864.35  5564.3 1893.31  5621.4 1912.03  5671.9 1919.84  5702.2 1921.52
#Mann= 10 ,-1 , 0
  4485.2     .07       0  4558.1      .1       0  4821.4     .07       0
  4904.3      .1       0  4981.1    .033       0  5041.9    .033       0
    5110    .033       0  5211.6     .07       0  5301.1    .035       0
  5564.3      .1       0
Bank Sta=5041.9,5110
XS Rating Curve= 0 ,0
Exp/Cntr=0.3,0.1

Type RM Length L Ch R = 1 ,34408   ,720,720,720
BEGIN DESCRIPTION:
South Fork Guadalupe River 48.0
END DESCRIPTION:
XS GIS Cut Line= 3
      1850385.24     13916201.23        1850175.       13915675.
        1850075.     13915174.98
#Sta/Elev= 30
  4441.8 1941.39  4508.8 1928.23  4545.4 1916.72  4640.8 1897.35  4646.2 1893.83
  4663.9 1890.74  4685.4 1881.24  4694.7 1872.75    4700 1871.27  4724.3 1850.78
  4748.5 1837.62  4768.9 1832.36  4802.4 1827.34  4861.7 1825.32  4876.2 1822.83
    4964 1824.29    4965 1822.49  4966.5 1821.49  5033.1 1822.49  5039.1 1826.06
  5090.1 1834.11  5161.4 1836.68  5273.6 1833.47  5288.1 1840.22  5304.2 1851.04
    5345 1872.69    5396 1896.01  5426.6 1899.85  5490.1 1901.97  5518.4 1902.88
#Mann= 7 ,-1 , 0
  4441.8      .1       0  4768.9     .07       0  4876.2    .094       0
    4965    .035       0  5033.1    .094       0  5288.1      .1       0
  5490.1     .07       0
Bank Sta=4965,5033.1
XS Rating Curve= 0 ,0
Exp/Cntr=0.3,0.1

Type RM Length L Ch R = 1 ,33688   ,538,538,538
BEGIN DESCRIPTION:
South Fork Guadalupe River 47.0
END DESCRIPTION:
XS GIS Cut Line= 3
        1850775.     13916025.04        1850775.       13915525.
      1850174.96     13915124.97
#Sta/Elev= 30
  4499.6 1949.04  4549.6 1941.04  4649.6 1932.99  4679.6 1928.92  4709.6 1921.26
  4749.6 1905.44  4759.6 1892.77  4769.6 1864.97  4804.4 1845.14  4829.6 1830.81
  4839.6 1827.97  4879.6 1828.32  4925.5 1822.47    4927 1821.47  4993.7 1822.47
  5094.3 1825.81  5121.3 1831.05  5185.6 1836.97  5274.6 1838.15  5403.8 1835.14
  5460.9 1831.36  5490.9 1832.44  5496.9 1838.54  5511.9 1848.74    5527 1862.78
    5533 1873.05    5569 1887.32  5576.8 1888.93  5620.1 1893.81  5720.8 1898.35
#Mann= 6 ,-1 , 0
  4499.6      .1       0  4804.4    .035       0  4925.5    .035       0
  4993.7    .035       0  5185.6      .1       0  5576.8     .07       0
Bank Sta=4925.5,4993.7
XS Rating Curve= 0 ,0
Exp/Cntr=0.3,0.1

Type RM Length L Ch R = 1 ,33150   ,421,421,421
BEGIN DESCRIPTION:
South Fork Guadalupe River 46.0
END DESCRIPTION:
XS GIS Cut Line= 3
        1851225.     13915725.02      1851163.97     13915285.01
      1850525.03     13914925.02
#Sta/Elev= 30
  4556.8 1918.34  4607.3 1916.87  4657.8 1910.61  4728.4 1906.24  4759.1 1898.42
  4768.8 1894.11  4778.9  1871.6    4789 1847.04  4812.9 1835.53  4819.3 1830.07
  4829.4 1828.19  4859.7 1828.71  4879.6 1824.18  4896.3 1822.63  4897.8 1821.63
  4964.5 1822.63  5008.4  1823.4  5093.7  1829.3  5148.6 1834.04  5309.8 1834.89
  5456.3  1833.2  5524.8 1830.76  5540.3 1831.16  5558.9 1831.03  5573.7 1834.13
  5580.6 1836.05  5602.2 1848.55  5623.9 1853.84  5711.5 1864.96  5734.4 1865.92
#Mann= 7 ,-1 , 0
  4556.8      .1       0  4759.1    .035       0  4896.3    .035       0
  4964.5    .035       0  5093.7      .1       0  5524.8    .035       0
  5540.3     .07       0
Bank Sta=4896.3,4964.5
XS Rating Curve= 0 ,0
Exp/Cntr=0.3,0.1

Type RM Length L Ch R = 1 ,32729   ,629,629,629
BEGIN DESCRIPTION:
South Fork Guadalupe River 45.1
END DESCRIPTION:
XS GIS Cut Line= 3
      1851488.93     13915565.31      1851542.73     13914794.01
      1851648.47     13914460.76
#Sta/Elev= 30
  4608.8 1908.88  4669.3 1905.64  4779.5 1889.67  4789.6  1874.9  4799.6 1869.86
  4809.6  1850.5    4823 1839.89  4829.6 1836.03  4859.7 1835.18  4869.7 1829.59
  4889.8 1823.36  4994.2 1822.24  4995.7 1821.24    5066 1822.24  5070.2  1824.6
  5140.4 1828.46  5197.3 1829.34  5240.6 1837.73  5302.8 1840.24  5414.5 1842.56
  5516.6 1843.63  5553.3 1844.34  5590.8 1847.62  5618.8 1861.49  5632.5 1866.66
  5643.2 1874.85  5664.2 1883.58    5670 1888.63  5707.5 1906.27  5731.6 1912.25
#Mann= 9 ,-1 , 0
  4608.8      .1       0    4823    .035       0  4994.2    .035       0
    5066    .035       0  5302.8    .035       0  5414.5     .07       0
  5516.6      .1       0  5553.3     .07       0  5618.8      .1       0
Bank Sta=4994.2,5066
XS Rating Curve= 0 ,0
Exp/Cntr=0.3,0.1

Type RM Length L Ch R = 1 ,32100   ,540,540,540
BEGIN DESCRIPTION:
South Fork Guadalupe River 45.0
END DESCRIPTION:
XS GIS Cut Line= 3
      1851624.98     13915475.01      1852028.04     13915164.59
      1852424.97     13914775.03
#Sta/Elev= 30
  4437.3 1896.49  4500.7 1889.97  4526.8 1884.09  4587.7 1856.51  4594.1 1851.62
    4627 1841.71  4687.4  1840.3  4693.7 1836.14  4701.9 1836.55  4708.2 1830.73
  4822.4 1825.84  4828.7 1821.93  4856.2 1822.25  4978.4 1821.92  4979.9 1820.92
  5050.2 1821.92  5056.7 1825.17  5073.8 1826.02  5191.1 1829.65  5205.3 1833.11
  5233.6 1847.86  5240.6 1865.33  5247.7 1861.18  5254.7 1884.32  5360.9 1944.88
  5367.9 1953.44  5403.3 1975.21  5417.4 1986.72    5481 2012.73  5502.2 2016.61
#Mann= 7 ,-1 , 0
  4437.3      .1       0  4526.8     .07       0    4627    .035       0
  4856.2    .033       0  4978.4    .033       0  5050.2    .033       0
  5073.8      .1       0
Bank Sta=4978.4,5050.2
XS Rating Curve= 0 ,0
Exp/Cntr=0.3,0.1

Type RM Length L Ch R = 1 ,31560   ,726,726,726
BEGIN DESCRIPTION:
South Fork Guadalupe River 44.0
END DESCRIPTION:
XS GIS Cut Line= 3
      1851925.03     13915674.99        1852525.       13915375.
      1852825.01     13914974.99
#Sta/Elev= 30
  4338.1 1892.04  4403.2 1883.61  4435.9 1873.74  4486.2 1850.57  4580.3 1843.12
  4601.2 1842.14  4695.8 1839.86  4726.6 1832.21  4793.7 1834.91  4860.3 1818.02
  4905.5 1820.76  4950.2 1816.53  4950.6 1809.46  4952.1 1808.46  5022.4 1809.46
  5095.3  1816.3  5122.1 1836.06  5151.6 1859.43  5158.9 1900.82  5172.4 1918.09
  5216.2 1944.36  5230.8 1956.45    5237 1970.63  5245.3 1970.82  5272.4 1998.19
  5280.8 1999.21    5287 2010.52  5322.4 2019.94  5416.2 2032.91  5508.9  2038.7
#Mann= 8 ,-1 , 0
  4338.1     .07       0  4403.2      .1       0  4580.3     .07       0
  4601.2    .035       0  4860.3     .07       0  4950.6     .05       0
  5022.4     .07       0  5122.1      .1       0
Bank Sta=4950.6,5022.4
XS Rating Curve= 0 ,0
Exp/Cntr=0.3,0.1

Type RM Length L Ch R = 1 ,30834   ,696,696,696
BEGIN DESCRIPTION:
South Fork Guadalupe River 43.0
END DESCRIPTION:
XS GIS Cut Line= 3
      1851925.04     13916324.99        1852925.       13915925.
        1853325.       13915625.
#Sta/Elev= 30
  3927.1    1918  4088.6 1895.71  4142.5 1893.03  4289.2 1857.73  4359.5 1851.04
  4493.7 1842.36  4576.3  1840.3  4695.8 1838.94  4725.4 1835.15  4788.7 1816.76
  4819.8 1816.44  4906.8  1813.7  4928.7 1813.76  4958.8 1807.19  4960.3 1806.19
  5030.6 1807.19  5046.8  1813.9  5061.4 1832.91  5067.6 1835.62    5076 1899.81
  5082.2 1913.19  5096.8 1924.67  5117.6 1947.26    5126 1961.55  5132.2 1965.21
  5140.6 1976.44  5146.8  1990.4  5211.4 2001.47  5437.9 2018.84  5504.1  2022.5
#Mann= 9 ,-1 , 0
  3927.1     .07       0  4359.5      .1       0  4493.7     .07       0
  4576.3    .035       0  4819.8     .07       0  4906.8    .035       0
  4958.8    .035       0  5030.6    .035       0  5437.9     .07       0
Bank Sta=4958.8,5030.6
XS Rating Curve= 0 ,0
Exp/Cntr=0.3,0.1

Type RM Length L Ch R = 1 ,30138   ,698,698,698
BEGIN DESCRIPTION:
South Fork Guadalupe River 42.0
END DESCRIPTION:
XS GIS Cut Line= 3
      1852075.02       13916575.        1853075.       13916575.
      1853375.01     13916174.98
#Sta/Elev= 30
  4004.6 1904.84  4105.5    1891  4174.6 1879.82  4264.6 1856.73  4294.6 1853.31
  4324.6 1845.17  4424.6 1840.73  4588.5 1838.35  4764.6  1835.8  4794.6 1830.89
  4843.3 1812.01  4864.6 1809.05  4941.9 1808.54    4976 1806.17  4977.5 1805.17
  5047.8 1806.17  5054.6 1810.51  5076.5 1814.76  5082.7 1819.42    5091 1820.28
  5111.9 1828.12  5118.1    1853  5126.5 1832.17  5132.7 1904.49  5147.3 1910.11
  5204.6 1927.84    5291 1947.33  5326.5 1952.67  5491.4 1957.87  5504.6 1958.18
#Mann= 8 ,-1 , 0
  4004.6      .1       0  4105.5     .07       0  4588.5    .035       0
  4843.3     .07       0  4941.9      .1       0    4976     .05       0
  5047.8      .1       0  5491.4     .07       0
Bank Sta=4976,5047.8
XS Rating Curve= 0 ,0
Exp/Cntr=0.3,0.1

Type RM Length L Ch R = 1 ,29440   ,716,716,716
BEGIN DESCRIPTION:
South Fork Guadalupe River 41.0
END DESCRIPTION:
XS GIS Cut Line= 3
      1852274.97     13917675.02        1853175.       13917175.
        1853675.       13917275.
#Sta/Elev= 30
  3962.2 1907.32  4078.9 1893.27  4138.4 1881.81  4197.9 1863.79  4257.4 1854.79
  4482.2 1848.17  4522.8 1846.95  4637.2 1830.64  4674.9 1830.59  4690.9 1822.18
  4722.7 1816.21  4756.1 1821.13  4772.2 1829.79  4785.9 1832.39  4831.6 1833.03
  4859.1 1831.36  4888.8 1819.46  4934.6 1809.38  5037.4  1806.4  5038.9  1805.4
  5109.3  1806.4  5175.4 1817.08  5199.8 1833.65  5226.4 1848.28  5236.6 1858.07
  5256.9 1889.21  5267.1 1896.41  5409.9 1939.99  5440.5 1953.63  5501.7 1968.97
#Mann= 6 ,-1 , 0
  3962.2      .1       0  4482.2    .035       0  4722.7      .1       0
  5037.4     .05       0  5109.3      .1       0  5199.8      .1       0
Bank Sta=5037.4,5109.3
XS Rating Curve= 0 ,0
Exp/Cntr=0.3,0.1

Type RM Length L Ch R = 1 ,28724   ,759,759,759
BEGIN DESCRIPTION:
South Fork Guadalupe River 40.0
END DESCRIPTION:
XS GIS Cut Line= 3
      1852375.02       13917725.        1853375.       13917725.
      1853775.02     13917424.99
#Sta/Elev= 30
  4004.8 1897.69  4094.8 1880.45  4174.8 1859.29  4377.6 1845.41  4474.8 1843.08
  4494.8 1840.65  4504.8 1836.26  4604.9 1833.26  4703.5 1831.34  4802.1 1826.99
  4844.8  1825.1  4874.8 1815.69  4900.7 1812.24  4924.8 1811.16  4944.8 1806.59
    4976 1806.37  4977.5 1805.37  5048.1 1806.37  5082.9 1807.09  5132.9 1815.74
  5168.3 1845.79  5176.7 1893.53  5197.5 1904.18  5212.1 1915.59  5218.3 1916.09
  5226.7 1921.68  5341.2  1960.9  5397.5 1972.45  5462.1 1991.62  5504.8 1996.03
#Mann= 8 ,-1 , 0
  4004.8      .1       0  4377.6    .035       0  4604.9     .07       0
  4703.5    .035       0  4802.1     .07       0  4900.7      .1       0
    4976     .05       0  5048.1      .1       0
Bank Sta=4976,5048.1
XS Rating Curve= 0 ,0
Exp/Cntr=0.3,0.1

Type RM Length L Ch R = 1 ,27965   ,529,529,529
BEGIN DESCRIPTION:
South Fork Guadalupe River 39.0
END DESCRIPTION:
XS GIS Cut Line= 3
      1852525.01       13918125.      1853400.93     13918276.92
      1854024.99       13918325.
#Sta/Elev= 30
  4078.5 1885.03  4105.8 1879.64  4110.9 1880.88  4165.5 1863.93    4180  1864.1
  4220.1  1853.5    4251 1849.67  4307.3 1848.24  4369.3 1845.61  4453.9 1842.16
  4545.4 1833.62  4613.4 1832.33  4712.8 1830.04  4819.4 1826.69  4880.7 1819.14
  4900.6 1816.49  4951.3 1815.56  4955.6 1807.39  4957.1 1806.39  5027.7 1807.39
  5142.4 1807.92  5208.2 1817.28  5232.3 1829.75  5262.4 1839.27  5267.7 1842.96
  5282.5  1846.5  5362.7 1882.37    5403 1896.72  5528.3 1919.04  5593.4 1927.49
#Mann= 9 ,-1 , 0
  4078.5      .1       0  4307.3     .07       0  4369.3    .035       0
  4613.4     .07       0  4712.8    .035       0  4880.7      .1       0
  4955.6     .05       0  5027.7      .1       0  5208.2      .1       0
Bank Sta=4955.6,5027.7
XS Rating Curve= 0 ,0
Exp/Cntr=0.3,0.1

Type RM Length L Ch R = 1 ,27436   ,716,716,716
BEGIN DESCRIPTION:
South Fork Guadalupe River 38.0
END DESCRIPTION:
XS GIS Cut Line= 3
      1852625.04       13918625.        1853625.       13918625.
      1854125.04     13918524.99
#Sta/Elev= 30
  3999.6 1897.09  4039.6 1890.47  4069.6 1889.82  4079.6 1886.51  4099.6 1874.79
  4120.9 1866.96  4219.6 1836.98  4259.6 1834.56  4416.6 1831.16  4579.6 1822.54
    4729 1816.98  4809.6 1814.28  4889.6 1807.09    4915 1806.73  4973.7 1805.99
  4975.2 1804.99  5045.8 1805.99  5050.5 1808.53  5081.1 1811.71  5101.5 1811.43
  5111.7 1813.62  5121.9 1818.28  5132.1 1829.02  5142.3 1835.02  5223.9 1877.75
  5254.5 1896.97  5305.5 1909.31  5387.1 1921.73  5438.1 1927.21  5509.5 1931.54
#Mann= 7 ,-1 , 0
  3999.6     .07       0  4120.9      .1       0  4416.6    .035       0
    4729     .07       0    4915      .1       0  4973.7     .05       0
  5045.8      .1       0
Bank Sta=4973.7,5045.8
XS Rating Curve= 0 ,0
Exp/Cntr=0.3,0.1

Type RM Length L Ch R = 1 ,26720   ,719,719,719
BEGIN DESCRIPTION:
South Fork Guadalupe River 37.0
END DESCRIPTION:
XS GIS Cut Line= 3
      1852875.01     13919724.99        1853675.       13919325.
      1854474.96       13919425.
#Sta/Elev= 30
  4105.5 1904.08  4186.5 1899.44  4231.3 1891.87  4239.6 1888.31    4248 1877.81
  4253.6    1856    4262 1847.41  4312.2 1821.16  4337.5 1816.61  4552.7 1820.52
  4884.5 1812.07  4955.2 1807.69    4961 1796.98  4962.5 1795.98  5033.2 1796.98
  5037.7 1800.36  5050.3  1801.4  5165.3 1801.99  5191.4 1802.57  5231.7 1824.17
  5365.2 1830.55    5421  1840.4  5436.3 1842.49  5483.6 1845.97  5526.5 1855.22
  5574.3 1868.78  5602.1 1880.68  5682.7 1906.81  5763.3 1926.75  5806.1 1933.43
#Mann= 8 ,-1 , 0
  4105.5      .1       0  4312.2    .035       0  4884.5     .07       0
    4961     .05       0  5033.2     .07       0  5165.3      .1       0
    5421     .07       0  5436.3      .1       0
Bank Sta=4961,5033.2
XS Rating Curve= 0 ,0
Exp/Cntr=0.3,0.1

Type RM Length L Ch R = 1 ,26001   ,687,687,687
BEGIN DESCRIPTION:
South Fork Guadalupe River 36.0
END DESCRIPTION:
XS GIS Cut Line= 3
        1853175.       13920275.        1853575.       13919975.
      1854574.96     13919575.01
#Sta/Elev= 30
    4500 1894.48  4528.1 1893.64  4542.7 1886.54    4550 1859.88  4557.3 1850.72
  4586.5 1834.13  4629.4 1819.51    4650 1812.51  4671.9 1811.35  4893.9 1810.54
  4907.3 1803.49  4928.1 1804.33  4935.8 1797.46  4937.3 1796.46    5008 1797.46
  5021.5 1799.92  5067.9 1798.71  5098.3 1798.84  5129.2 1805.55  5146.8 1820.41
  5152.1  1819.7    5171 1826.88  5588.3 1825.43  5700.1 1833.15  5732.4 1838.42
  5757.5 1846.87  5883.2 1900.99  5954.5 1924.29  6023.2 1937.62    6077 1941.22
#Mann= 8 ,-1 , 0
    4500      .1       0  4629.4    .035       0  4893.9     .07       0
  4935.8     .05       0    5008     .07       0  5067.9      .1       0
  5588.3     .07       0  5757.5      .1       0
Bank Sta=4935.8,5008
XS Rating Curve= 0 ,0
Exp/Cntr=0.3,0.1

Type RM Length L Ch R = 1 ,25314   ,667,667,667
BEGIN DESCRIPTION:
South Fork Guadalupe River 35.0
END DESCRIPTION:
XS GIS Cut Line= 3
      1853325.03     13920974.97        1853625.       13920575.
      1854625.01     13919774.99
#Sta/Elev= 30
  4500.6 1909.26  4578.7 1894.64  4643.3 1872.28  4659.4 1861.22  4672.4 1855.86
  4693.3 1852.52  4707.8 1843.02  4714.1 1843.14    4737 1828.24  4757.8 1828.08
  4772.4 1822.86  4778.7  1816.9  4793.3  1810.4  4906.5 1797.12  4941.2 1796.97
  4957.1 1796.49  4958.6 1795.49  5029.4 1796.49    5051    1800  5092.6 1799.82
  5121.4 1811.31  5135.8 1824.12  5164.6 1826.32  5491.2 1825.44  5668.9 1821.17
  5790.5 1824.71  5953.8 1838.54  6017.9 1853.52  6217.2 1925.64  6281.2 1937.91
#Mann= 6 ,-1 , 0
  4500.6      .1       0  4659.4    .035       0  4906.5     .07       0
  4941.2      .1       0  4957.1     .05       0  5029.4      .1       0
Bank Sta=4957.1,5029.4
XS Rating Curve= 0 ,0
Exp/Cntr=0.3,0.1

Type RM Length L Ch R = 1 ,24647   ,587,587,587
BEGIN DESCRIPTION:
South Fork Guadalupe River 34.0
END DESCRIPTION:
XS GIS Cut Line= 3
      1853474.97     13921375.02        1853875.       13921075.
      1854557.16     13920021.51
#Sta/Elev= 30
  4505.2 1925.49  4600.3 1916.36  4688.1 1903.42  4741.7 1894.47  4796.9  1877.1
  4805.2 1872.54  4812.5    1842  4841.7 1826.77  4868.8 1807.13  4877.1  1803.9
  4890.7 1803.77  4905.2 1803.58  4927.1 1796.74  4976.7 1796.54  4978.2 1795.54
    5049 1796.54  5049.1 1798.41  5068.4 1799.72  5120.1 1800.82    5172 1810.73
  5215.3 1823.52  5562.8 1823.65  5734.9 1817.22  6076.5  1830.5  6133.9  1844.9
  6206.4 1870.18  6212.4 1874.09  6242.7 1882.33  6248.7 1886.42  6260.3 1887.47
#Mann= 8 ,-1 , 0
  4505.2      .1       0  4600.3     .07       0  4688.1    .035       0
  4890.7      .1       0  4976.7     .05       0    5049      .1       0
  5068.4    .033       0  5120.1      .1       0
Bank Sta=4976.7,5049
XS Rating Curve= 0 ,0
Exp/Cntr=0.3,0.1

Type RM Length L Ch R = 1 ,24060   ,837,837,837
BEGIN DESCRIPTION:
South Fork Guadalupe River 33.0
END DESCRIPTION:
XS GIS Cut Line= 3
      1853725.02       13921525.      1854107.29     13921532.03
      1855225.04     13921124.98
#Sta/Elev= 30
  4559.7 1905.52  4670.7  1888.1  4709.7 1877.82  4749.7 1843.73  4799.7 1812.71
  4809.7 1810.08  4839.7 1809.62  4849.7 1807.47  4859.7 1800.32  4924.7 1796.53
  4926.2 1795.53    4997 1796.53  5068.8  1799.4  5141.8 1797.47  5185.7 1802.81
  5201.2 1801.85  5241.6 1797.86  5258.9  1804.3  5286.7 1804.48  5302.7 1804.48
  5353.2 1816.64    5499 1818.13  5812.3 1820.29  5885.3 1826.11  5912.4 1832.05
  5918.7 1835.93  5993.2 1858.18  6055.1 1882.15  6099.6 1895.86  6131.6 1899.78
#Mann= 8 ,-1 , 0
  4559.7      .1       0  4670.7    .035       0  4924.7     .05       0
    4997    .035       0  5201.2    .035       0  5286.7      .1       0
    5499     .07       0  5885.3      .1       0
Bank Sta=4924.7,4997
XS Rating Curve= 0 ,0
Exp/Cntr=0.3,0.1
