HEC-RAS study Stream0095.prj: Stream0095 Base Level Engineering

--- Stream0095.g01 (geometry) --- (continued)

Type RM Length L Ch R = 1,29580,587,587,587
BEGIN DESCRIPTION:
Stream0095 51.0
END DESCRIPTION:
XS GIS Cut Line= 3
      1776025.01     13911274.97      1776175.00     13910875.00
      1776724.98     13910625.01
#Sta/Elev= 30
  4574.1 2235.50  4583.9 2234.82  4589.2 2235.52  4614.1 2233.34  4619.5 2233.90
  4669.3 2230.95  4674.6 2231.52  4712.7 2228.03  4798.4 2220.29  4845.5 2215.23
  4862.4 2212.16  4894.5 2209.23  4915.8 2203.39  4925.6 2190.41  4931.0 2184.40
  4937.2 2179.63  4947.9 2177.55  4951.0 2174.98  4951.5 2174.48  4971.4 2174.98
  5004.0 2177.63  5010.1 2179.01  5038.2 2180.49  5078.2 2182.65  5177.0 2182.67
  5251.7 2186.19  5257.2 2185.42  5297.9 2186.16  5407.7 2193.96  5605.4 2200.94
#Mann=5,-1,0
  4574.1     0.1       0  4712.7    0.07       0  4951.0    0.05       0
  4971.4    0.07       0  5038.2     0.1       0
Bank Sta=4951,4971.4
Exp/Cntr=0.3,0.1

Type RM Length L Ch R = 1,28993,562,562,562
BEGIN DESCRIPTION:
Stream0095 50.0
END DESCRIPTION:
XS GIS Cut Line= 3
      1776225.01     13911475.00      1776575.00     13911275.00
      1776825.02     13910724.96
#Sta/Elev= 30
  4601.3 2239.23  4674.0 2238.78  4733.0 2234.57  4762.5 2227.60  4785.6 2225.21
  4792.0 2223.36  4813.6 2220.37  4829.5 2217.24  4835.2 2217.36  4843.2 2215.29
  4866.2 2211.99  4878.4 2209.31  4910.1 2200.76  4923.8 2195.91  4931.7 2194.43
  4937.5 2191.04  4946.8 2189.57  4953.3 2183.96  4959.1 2181.19  4974.9 2176.10
  4991.3 2174.12  4991.8 2173.62  5011.7 2174.12  5036.3 2175.61  5111.0 2183.27
  5214.2 2189.04  5381.2 2192.94  5496.5 2196.43  5502.0 2197.21  5608.6 2199.93
#Mann=3,-1,0
  4601.3     0.1       0  4991.3    0.05       0  5011.7     0.1       0
Bank Sta=4991.3,5011.7
Exp/Cntr=0.3,0.1

Type RM Length L Ch R = 1,28431,556,556,556
BEGIN DESCRIPTION:
Stream0095 49.0
END DESCRIPTION:
XS GIS Cut Line= 3
      1776624.97     13911725.01      1777025.00     13911525.00
      1777175.00     13910925.01
#Sta/Elev= 30
  4558.6 2224.72  4595.0 2221.78  4634.1 2215.73  4678.8 2211.85  4706.8 2207.48
  4745.9 2204.31  4751.5 2202.69  4813.0 2196.66  4818.6 2195.01  4835.3 2194.46
  4840.9 2192.94  4885.7 2189.15  4902.4 2188.64  4908.0 2186.35  4924.8 2186.02
  4930.4 2182.18  4947.1 2179.88  4952.7 2176.47  4969.5 2175.11  4973.3 2173.01
  4973.8 2172.51  4993.7 2173.01  4997.5 2174.33  5016.2 2175.24  5023.9 2176.67
  5065.1 2177.52  5098.6 2180.71  5235.2 2186.15  5271.3 2188.78  5624.3 2198.61
#Mann=3,-1,0
  4558.6     0.1       0  4973.3    0.05       0  4993.7     0.1       0
Bank Sta=4973.3,4993.7
Exp/Cntr=0.3,0.1

Type RM Length L Ch R = 1,27875,559,559,559
BEGIN DESCRIPTION:
Stream0095 48.0
END DESCRIPTION:
XS GIS Cut Line= 3
      1777875.01     13911675.01      1777525.00     13911475.00
      1777375.00     13910925.01
#Sta/Elev= 30
  4596.9 2223.17  4648.0 2222.63  4728.6 2219.73  4787.7 2215.67  4825.1 2211.91
  4830.9 2209.96  4861.8 2205.89  4868.3 2204.51  4874.1 2201.64  4884.1 2201.33
  4889.9 2198.75  4896.4 2197.15  4905.7 2196.10  4911.5 2192.37  4927.3 2188.13
  4933.1 2183.91  4954.7 2175.43  4964.8 2174.54  4976.1 2171.06  4976.6 2170.56
  4996.5 2171.06  4997.1 2171.83  5031.1 2174.03  5062.2 2179.09  5114.0 2179.60
  5136.5 2181.59  5250.5 2183.43  5279.9 2186.82  5331.7 2190.13  5570.1 2197.37
#Mann=3,-1,0
  4596.9     0.1       0  4976.1    0.05       0  4996.5     0.1       0
Bank Sta=4976.1,4996.5
Exp/Cntr=0.3,0.1

Type RM Length L Ch R = 1,27316,590,590,590
BEGIN DESCRIPTION:
Stream0095 47.0
END DESCRIPTION:
XS GIS Cut Line= 3
      1777975.00     13911575.01      1777975.00     13911175.00
      1777525.04     13910875.02
#Sta/Elev= 30
  4600.3 2224.34  4680.3 2222.04  4760.3 2217.24  4820.3 2212.99  4880.3 2207.29
  4900.3 2203.70  4940.3 2195.02  4950.3 2190.61  4960.3 2181.19  4970.3 2176.16
  4980.3 2173.14  4997.8 2170.03  5012.6 2169.07  5013.1 2168.57  5032.6 2168.57
  5033.1 2169.07  5043.9 2171.28  5064.9 2172.90  5085.9 2173.47  5101.0 2175.87
  5108.5 2177.78  5137.0 2178.47  5167.1 2180.91  5173.1 2181.96  5188.1 2182.37
  5230.2 2185.32  5311.3 2188.34  5353.4 2189.13  5440.5 2192.99  5541.1 2195.12
#Mann=3,-1,0
  4600.3     0.1       0  5012.6    0.05       0  5033.1     0.1       0
Bank Sta=5012.6,5033.1
Exp/Cntr=0.3,0.1

Type RM Length L Ch R = 1,26726,1073,1073,1073
BEGIN DESCRIPTION:
Stream0095 46.0
END DESCRIPTION:
XS GIS Cut Line= 4
      1778395.03     13911330.60      1778391.54     13910968.98
      1778325.00     13910725.00      1777575.00     13910425.00
#Sta/Elev= 30
  4381.3 2201.16  4666.9 2188.48  4736.9 2186.42  4778.2 2183.41  4859.4 2179.99
  4871.4 2178.72  4892.2 2177.94  4933.6 2174.18  4944.0 2172.34  4983.0 2171.09
  4983.5 2170.59  5003.5 2171.09  5028.1 2171.50  5040.3 2173.14  5064.5 2172.43
  5125.1 2178.09  5142.6 2178.80  5196.4 2179.10  5232.8 2180.38  5243.5 2181.41
  5279.9 2182.69  5328.4 2186.61  5372.8 2188.59  5405.1 2188.70  5465.7 2191.09
  5519.5 2191.51  5543.8 2192.68  5616.4 2194.13  5771.3 2196.30  5803.6 2197.54
#Mann=4,-1,0
  4381.3     0.1       0  4983.0    0.05       0  5003.5     0.1       0
  5616.4    0.07       0
Bank Sta=4983,5003.5
Exp/Cntr=0.3,0.1

Type RM Length L Ch R = 1,25653,556,556,556
BEGIN DESCRIPTION:
Stream0095 45.0
END DESCRIPTION:
XS GIS Cut Line= 4
      1778693.75     13910994.10      1778875.00     13910609.34
      1778875.00     13909975.00      1778524.97     13909774.98
#Sta/Elev= 30
  3940.3 2190.65  4052.1 2189.71  4285.5 2190.57  4331.1 2190.08  4410.0 2187.60
  4636.1 2183.23  4734.4 2180.46  4820.0 2179.00  4870.0 2177.22  4900.0 2173.79
  4920.0 2172.75  4960.0 2167.46  4990.0 2166.40  4997.6 2164.77  4998.1 2164.27
  5017.7 2164.27  5018.2 2164.77  5029.5 2166.76  5045.3 2167.72  5051.1 2170.34
  5066.9 2173.96  5072.7 2177.48  5094.3 2180.55  5110.1 2181.27  5206.6 2189.00
  5228.1 2192.20  5287.2 2196.77  5367.8 2205.53  5380.0 2207.42  5403.1 2208.91
#Mann=5,-1,0
  3940.3     0.1       0  4636.1    0.07       0  4734.4     0.1       0
  4997.6    0.05       0  5018.2     0.1       0
Bank Sta=4997.6,5018.2
Exp/Cntr=0.3,0.1

Type RM Length L Ch R = 1,25097,445,445,445
BEGIN DESCRIPTION:
Stream0095 44.0
END DESCRIPTION:
XS GIS Cut Line= 3
      1778719.71     13911002.92      1779375.00     13909975.00
      1779474.99     13909575.03
#Sta/Elev= 30
  3780.6 2190.39  3849.3 2189.73  3876.5 2190.33  4006.9 2189.71  4094.9 2190.67
  4167.7 2190.04  4325.1 2186.31  4419.0 2185.45  4434.3 2184.17  4557.8 2183.25
  4689.0 2182.26  4798.1 2177.03  4860.1 2175.63  4882.8 2174.28  4919.2 2170.51
  4949.7 2165.33  4992.0 2163.59  4999.5 2161.17  5000.0 2160.67  5020.3 2161.17
  5022.8 2165.77  5030.5 2170.67  5040.9 2175.32  5064.0 2180.00  5092.4 2188.33
  5146.5 2192.70  5216.1 2195.89  5306.3 2202.84  5370.7 2205.84  5411.9 2209.07
#Mann=5,-1,0
  3780.6     0.1       0  4557.8    0.07       0  4798.1     0.1       0
  4999.5    0.05       0  5020.3     0.1       0
Bank Sta=4999.5,5020.3
Exp/Cntr=0.3,0.1

Type RM Length L Ch R = 1,24652,394,394,394
BEGIN DESCRIPTION:
Stream0095 43.0
END DESCRIPTION:
XS GIS Cut Line= 4
      1778874.63     13910800.07      1779069.04     13910554.39
      1779718.11     13910250.69      1779842.31     13909348.19
#Sta/Elev= 30
  3983.1 2189.99  4115.7 2189.65  4279.2 2186.10  4369.2 2182.83  4495.9 2182.64
  4564.4 2180.26  4758.1 2177.98  4781.0 2177.21  4826.6 2173.45  4877.8 2172.33
  4900.7 2170.52  4940.8 2164.38  4976.4 2163.84  4992.0 2163.14  4998.1 2161.86
  4998.6 2161.36  5018.9 2161.86  5049.0 2169.73  5069.2 2172.08  5097.3 2177.34
  5129.8 2180.11  5311.5 2188.92  5395.5 2194.28  5442.7 2194.70  5573.9 2200.22
  5683.5 2207.38  5760.5 2210.34  5796.0 2212.81  5856.6 2215.39  5924.0 2220.68
#Mann=3,-1,0
  3983.1     0.1       0  4998.1    0.05       0  5018.9     0.1       0
Bank Sta=4998.1,5018.9
Exp/Cntr=0.3,0.1

Type RM Length L Ch R = 1,24258,338,338,338
BEGIN DESCRIPTION:
Mapping XS 5bc4179a
END DESCRIPTION:
XS GIS Cut Line= 4
      1778974.45     13910730.92      1779119.98     13910569.82
      1779604.99     13910536.53      1779924.47     13910909.83
#Sta/Elev= 30
  4255.3 2188.58  4477.4 2183.09  4619.3 2181.68  4698.0 2177.62  4858.3 2172.53
  4888.4 2170.49  4905.7 2168.08  4910.7 2169.49  4918.5 2168.50  4938.5 2165.31
  4956.1 2161.12  4971.3 2159.40  4988.6 2155.23  4989.1 2154.73  5011.1 2155.23
  5021.8 2158.88  5035.5 2167.84  5042.6 2177.07  5063.5 2189.81  5077.8 2191.00
  5120.6 2201.04  5163.4 2206.77  5227.0 2213.53  5305.0 2216.49  5319.2 2218.21
  5382.9 2221.26  5425.7 2225.96  5432.3 2224.87  5440.0 2226.48  5449.9 2225.66
#Mann=3,-1,0
  4255.3     0.1       0  4988.6    0.05       0  5011.1     0.1       0
Bank Sta=4988.6,5011.1
Exp/Cntr=0.3,0.1

Type RM Length L Ch R = 1,23920,542,542,542
BEGIN DESCRIPTION:
Stream0095 42.0
END DESCRIPTION:
XS GIS Cut Line= 3
      1779025.01     13910775.00      1779425.00     13910825.00
      1779825.00     13910975.00
#Sta/Elev= 30
  4596.9 2186.64  4727.9 2179.85  4758.1 2179.50  4795.9 2176.87  4828.7 2175.89
  4869.0 2171.09  4889.1 2166.31  4899.2 2164.91  4919.4 2164.53  4939.5 2162.12
  4969.8 2161.35  4978.7 2160.11  4979.2 2159.61  5001.2 2160.11  5032.0 2161.09
  5045.4 2163.04  5064.1 2170.30  5070.3 2173.69  5085.4 2177.30  5125.5 2189.14
  5210.9 2206.15  5216.3 2206.15  5241.2 2211.36  5271.5 2214.01  5296.4 2219.00
  5301.7 2218.70  5320.4 2221.94  5326.6 2224.27  5373.8 2228.80  5427.2 2231.09
#Mann=3,-1,0
  4596.9     0.1       0  4978.7    0.05       0  5001.2     0.1       0
Bank Sta=4978.7,5001.2
Exp/Cntr=0.3,0.1

Type RM Length L Ch R = 1,23378,570,570,570
BEGIN DESCRIPTION:
Stream0095 41.0
END DESCRIPTION:
XS GIS Cut Line= 3
      1778774.97     13911275.00      1779175.00     13911275.00
      1779874.98     13911125.00
#Sta/Elev= 30
  4600.3 2190.97  4650.3 2189.26  4710.3 2185.24  4830.3 2182.43  4870.3 2180.02
  4940.3 2170.01  4970.3 2161.39  4979.0 2157.55  4979.5 2157.05  5001.6 2157.55
  5041.2 2161.26  5112.8 2163.94  5118.8 2165.44  5133.3 2165.85  5163.1 2169.14
  5168.2 2168.52  5204.9 2171.52  5212.5 2173.12  5245.8 2175.50  5306.3 2182.92
  5360.8 2187.66  5399.2 2192.71  5405.1 2194.60  5504.0 2207.32  5548.3 2214.65
  5583.3 2217.85  5603.7 2221.43  5634.4 2224.52  5685.5 2232.93  5716.2 2235.47
#Mann=3,-1,0
  4600.3     0.1       0  4979.0    0.05       0  5001.6     0.1       0
Bank Sta=4979,5001.6
Exp/Cntr=0.3,0.1

Type RM Length L Ch R = 1,22808,541,541,541
BEGIN DESCRIPTION:
Stream0095 40.0
END DESCRIPTION:
XS GIS Cut Line= 3
      1778625.00     13911575.00      1779068.69     13911827.21
      1779830.43     13911978.59
#Sta/Elev= 30
  4593.1 2196.60  4638.5 2195.91  4644.3 2195.01  4696.6 2193.27  4746.6 2189.11
  4821.6 2181.31  4857.7 2179.00  4870.6 2176.49  4945.6 2168.62  4951.3 2167.75
  4967.2 2162.67  4973.0 2161.63  4988.8 2160.85  5007.4 2158.44  5007.9 2157.94
  5030.0 2158.44  5053.7 2159.87  5103.5 2160.21  5121.5 2161.43  5150.7 2165.53
  5181.3 2168.20  5283.2 2175.02  5479.5 2184.81  5609.5 2190.34  5632.9 2191.88
  5650.3 2194.40  5684.0 2197.21  5691.0 2198.72  5742.0 2203.12  5880.1 2210.27
#Mann=3,-1,0
  4593.1     0.1       0  5007.4    0.05       0  5030.0     0.1       0
Bank Sta=5007.4,5030
Exp/Cntr=0.3,0.1

Type RM Length L Ch R = 1,22267,534,534,534
BEGIN DESCRIPTION:
Stream0095 39.0
END DESCRIPTION:
XS GIS Cut Line= 3
      1778275.00     13911825.00      1778925.00     13912275.00
      1779224.97     13912624.96
#Sta/Elev= 30
  4214.1 2207.71  4242.5 2206.46  4329.0 2198.98  4400.6 2194.47  4466.1 2187.90
  4530.3 2184.37  4588.4 2178.35  4603.3 2177.82  4645.2 2173.44  4688.4 2170.33
  4773.6 2166.44  4818.2 2162.78  4955.3 2160.03  4982.4 2157.55  4990.3 2155.66
  4990.8 2155.16  5013.0 2155.66  5018.4 2161.07  5032.7 2167.13  5046.9 2170.30
  5061.2 2172.07  5181.9 2178.24  5239.0 2179.70  5253.3 2181.79  5259.9 2181.08
  5288.4 2181.68  5366.3 2186.74  5380.6 2188.52  5444.2 2192.70  5465.6 2195.11
#Mann=3,-1,0
  4214.1     0.1       0  4990.3    0.05       0  5013.0     0.1       0
Bank Sta=4990.3,5013
Exp/Cntr=0.3,0.1

Type RM Length L Ch R = 1,21733,560,560,560
BEGIN DESCRIPTION:
Stream0095 38.0
END DESCRIPTION:
XS GIS Cut Line= 3
      1778075.01     13911875.01      1778625.00     13912675.00
      1779124.98     13912775.00
#Sta/Elev= 30
  4029.2 2215.16  4129.3 2207.48  4144.2 2207.15  4323.5 2190.04  4490.3 2179.40
  4625.2 2173.24  4669.9 2170.22  4696.9 2166.81  4744.8 2165.57  4777.4 2166.65
  4792.3 2166.56  4798.4 2165.30  4842.3 2166.03  4885.0 2164.77  4914.8 2162.09
  4941.8 2156.78  4971.6 2153.90  4981.2 2151.89  4981.7 2151.39  5003.9 2151.89
  5020.4 2152.96  5030.6 2155.45  5051.0 2160.80  5061.2 2165.13  5081.6 2171.44
  5112.2 2174.80  5132.6 2176.46  5356.9 2181.60  5469.1 2189.20  5509.9 2193.33
#Mann=4,-1,0
  4029.2     0.1       0  4744.8    0.07       0  4981.2    0.05       0
  5003.9     0.1       0
Bank Sta=4981.2,5003.9
Exp/Cntr=0.3,0.1

Type RM Length L Ch R = 1,21173,549,549,549
BEGIN DESCRIPTION:
Stream0095 37.0
END DESCRIPTION:
XS GIS Cut Line= 3
      1777924.95     13913125.00      1778325.00     13913125.00
      1778825.05     13913024.99
#Sta/Elev= 30
  4600.3 2188.90  4610.3 2188.20  4620.3 2186.25  4640.3 2184.80  4670.3 2183.02
  4680.3 2182.99  4754.2 2178.11  4770.3 2177.52  4790.3 2175.91  4850.3 2170.21
  4890.3 2165.64  4940.3 2161.52  4960.3 2157.08  4970.3 2155.69  4978.9 2153.60
  4979.4 2153.10  5001.3 2153.10  5001.8 2153.60  5010.5 2154.51  5020.7 2154.18
  5041.1 2155.29  5092.1 2155.42  5143.1 2157.89  5163.5 2160.09  5183.9 2163.29
  5296.1 2173.90  5336.9 2175.72  5408.3 2177.04  5428.7 2177.91  5510.3 2179.83
#Mann=4,-1,0
  4600.3    0.07       0  4754.2     0.1       0  4978.9    0.05       0
  5001.8     0.1       0
Bank Sta=4978.9,5001.8
Exp/Cntr=0.3,0.1

Type RM Length L Ch R = 1,20624,564,564,564
BEGIN DESCRIPTION:
Stream0095 36.0
END DESCRIPTION:
XS GIS Cut Line= 3
      1777925.01     13913425.01      1778275.00     13913625.00
      1778774.99     13913425.01
#Sta/Elev= 30
  4592.8 2180.82  4628.1 2179.14  4767.7 2175.83  4795.0 2174.50  4857.7 2170.89
  4880.0 2168.95  4929.0 2166.89  4944.8 2164.66  4950.5 2165.25  4960.6 2163.87
  4966.4 2164.90  4982.2 2154.40  4988.0 2155.32  4993.0 2152.90  4998.6 2152.90
  5006.0 2149.78  5006.5 2149.28  5028.4 2149.28  5028.9 2149.78  5034.9 2152.05
  5040.3 2151.96  5071.3 2156.16  5113.0 2157.08  5142.6 2159.01  5211.3 2161.09
  5250.3 2164.98  5296.0 2167.63  5411.9 2172.28  5502.1 2175.25  5534.4 2175.57
#Mann=5,-1,0
  4592.8    0.07       0  4795.0     0.1       0  5006.0    0.05       0
  5028.9     0.1       0  5296.0    0.07       0
Bank Sta=5006,5028.9
Exp/Cntr=0.3,0.1

Type RM Length L Ch R = 1,20060,501,501,501
BEGIN DESCRIPTION:
Stream0095 35.0
END DESCRIPTION:
XS GIS Cut Line= 3
      1778575.00     13914474.98      1778575.00     13914075.00
      1778925.00     13913875.00
#Sta/Elev= 30
  4599.8 2199.03  4639.8 2194.75  4659.8 2191.79  4689.8 2189.51  4759.8 2173.69
  4789.8 2168.88  4799.8 2166.68  4839.8 2161.34  4859.8 2157.92  4889.8 2155.71
  4939.8 2150.20  4968.2 2149.28  4968.7 2148.78  4990.8 2148.78  4991.3 2149.28
  4997.3 2150.03  5029.3 2150.07  5045.1 2150.97  5057.4 2154.39  5072.5 2156.53
  5094.1 2158.84  5103.4 2158.63  5125.8 2160.39  5163.6 2164.20  5228.0 2170.00
  5271.2 2173.02  5287.0 2173.42  5308.6 2175.36  5352.7 2175.57  5402.9 2175.90
#Mann=5,-1,0
  4599.8     0.1       0  4968.2    0.05       0  4991.3     0.1       0
  5163.6   0.035       0  5352.7    0.07       0
Bank Sta=4968.2,4991.3
Exp/Cntr=0.3,0.1

Type RM Length L Ch R = 1,19559,590,590,590
BEGIN DESCRIPTION:
Stream0095 34.0
END DESCRIPTION:
XS GIS Cut Line= 3
      1778624.98     13914575.01      1778929.27     13914396.86
      1779080.35     13913702.71
#Sta/Elev= 30
  4623.9 2204.69  4694.6 2204.63  4749.1 2204.06  4796.6 2201.17  4866.4 2196.92
  4872.2 2195.23  4887.9 2195.68  4893.7 2193.34  4925.1 2191.31  4930.9 2184.45
  4946.5 2181.54  4952.3 2172.64  4968.0 2171.60  4973.4 2163.07  4981.7 2163.48
  4988.6 2151.49  4998.9 2147.22  5019.3 2141.85  5019.8 2141.35  5042.4 2141.85
  5050.0 2146.15  5069.7 2151.43  5098.9 2153.21  5131.9 2155.38  5167.9 2160.76
  5204.7 2162.97  5375.1 2171.64  5438.4 2174.06  5561.8 2176.48  5686.9 2177.34
#Mann=9,-1,0
  4623.9    0.07       0  4694.6     0.1       0  4796.6    0.07       0
  5019.3    0.05       0  5042.4    0.07       0  5098.9     0.1       0
  5204.7   0.035       0  5375.1    0.07       0  5438.4   0.035       0
Bank Sta=5019.3,5042.4
Exp/Cntr=0.3,0.1

Type RM Length L Ch R = 1,18969,706,706,706
BEGIN DESCRIPTION:
Stream0095 33.0
END DESCRIPTION:
XS GIS Cut Line= 3
      1779275.02     13914674.97      1779475.00     13914325.00
      1779289.45     13913678.06
#Sta/Elev= 30
  4596.9 2186.97  4700.5 2184.35  4744.4 2182.15  4809.2 2178.24  4852.4 2174.45
  4868.2 2171.93  4889.8 2171.00  4905.7 2166.83  4919.4 2164.62  4927.3 2161.13
  4933.0 2161.59  4948.9 2152.33  4954.6 2153.60  4964.7 2149.08  4970.5 2149.57
  4976.9 2146.06  4985.5 2142.83  4986.0 2142.33  5008.6 2142.83  5016.8 2145.25
  5022.0 2145.35  5031.2 2147.34  5055.8 2147.94  5151.0 2156.80  5240.1 2162.15
  5295.6 2163.79  5491.9 2174.26  5603.5 2176.73  5652.6 2176.55  5673.0 2176.91
#Mann=6,-1,0
  4596.9     0.1       0  4985.5    0.05       0  5008.6     0.1       0
  5151.0    0.07       0  5295.6   0.035       0  5652.6    0.07       0
Bank Sta=4985.5,5008.6
Exp/Cntr=0.3,0.1

Type RM Length L Ch R = 1,18263,451,451,451
BEGIN DESCRIPTION:
Stream0095 32.0
END DESCRIPTION:
XS GIS Cut Line= 3
      1779825.02     13914574.98      1780087.31     13914264.33
      1780324.99     13913875.02
#Sta/Elev= 30
  4535.4 2171.29  4659.3 2165.16  4776.6 2158.99  4819.4 2155.36  4848.0 2151.07
  4918.3 2147.81  4926.1 2146.49  4944.5 2145.64  4947.1 2142.78  4952.9 2144.29
  4962.5 2142.35  4983.9 2141.85  4999.3 2138.79  4999.8 2137.46  5000.3 2136.96
  5023.1 2137.46  5026.5 2141.28  5034.9 2145.78  5041.6 2150.90  5057.4 2158.20
  5063.2 2162.39  5078.7 2168.32  5105.9 2174.45  5121.3 2176.78  5128.6 2180.01
  5158.1 2186.60  5204.2 2191.62  5295.6 2201.68  5353.6 2206.58  5398.1 2208.78
#Mann=6,-1,0
  4535.4    0.07       0  4659.3     0.1       0  4999.8    0.05       0
  5023.1     0.1       0  5041.6     0.1       0  5204.2    0.07       0
Bank Sta=4999.8,5023.1
Exp/Cntr=0.3,0.1

Type RM Length L Ch R = 1,17812,551,551,551
BEGIN DESCRIPTION:
Stream0095 31.0
END DESCRIPTION:
XS GIS Cut Line= 3
      1780075.03     13914724.98      1780425.00     13914525.00
      1780625.00     13914174.99
#Sta/Elev= 30
  4600.9 2169.93  4638.8 2169.64  4658.3 2169.11  4748.4 2161.65  4775.8 2160.67
  4865.8 2153.95  4888.1 2151.27  4946.4 2139.86  4958.6 2134.89  4974.5 2132.87
  4978.7 2130.06  4979.2 2129.56  5002.0 2130.06  5004.0 2135.10  5006.9 2135.10
  5027.0 2146.90  5033.5 2153.14  5039.3 2162.42  5049.3 2165.96  5055.1 2170.80
  5070.9 2176.24  5084.6 2183.84  5098.3 2189.46  5114.1 2189.67  5135.7 2193.95
  5151.5 2195.42  5178.9 2200.15  5194.7 2201.34  5237.9 2207.81  5407.1 2217.51
#Mann=5,-1,0
  4600.9     0.1       0  4638.8    0.07       0  4658.3     0.1       0
  4978.7    0.05       0  5002.0     0.1       0
Bank Sta=4978.7,5002
Exp/Cntr=0.3,0.1

Type RM Length L Ch R = 1,17261,566,566,566
BEGIN DESCRIPTION:
Stream0095 30.0
END DESCRIPTION:
XS GIS Cut Line= 3
      1780174.95     13914924.99      1780575.00     13915025.00
      1780925.03     13914824.99
#Sta/Elev= 30
  4587.6 2169.68  4659.8 2166.00  4811.8 2153.65  4845.3 2152.15  4876.3 2148.16
  4894.3 2144.08  4935.5 2138.85  4940.7 2139.33  4978.0 2131.86  4978.5 2131.36
  5001.3 2131.86  5007.9 2134.89  5013.6 2135.38  5023.0 2138.86  5035.2 2153.74
  5045.3 2161.09  5051.1 2163.44  5057.5 2169.53  5066.9 2173.37  5072.7 2174.00
  5088.5 2179.58  5094.3 2180.61  5110.1 2186.73  5131.7 2188.70  5151.4 2191.94
  5184.2 2196.37  5218.8 2202.79  5249.7 2205.43  5276.6 2206.10  5403.1 2206.07
#Mann=5,-1,0
  4587.6     0.1       0  4978.0    0.05       0  5001.3     0.1       0
  5151.4    0.07       0  5276.6     0.1       0
Bank Sta=4978,5001.3
Exp/Cntr=0.3,0.1

Type RM Length L Ch R = 1,16695,546,546,546
BEGIN DESCRIPTION:
Stream0095 29.0
END DESCRIPTION:
XS GIS Cut Line= 3
      1780125.00     13915575.00      1780525.00     13915575.00
      1780874.99     13915375.01
#Sta/Elev= 30
  4600.0 2165.59  4650.0 2162.29  4710.0 2155.98  4790.0 2152.20  4810.0 2149.49
  4890.0 2144.34  4920.0 2141.04  4940.0 2136.97  4980.0 2134.77  4985.8 2130.32
  4986.3 2129.82  5009.3 2130.32  5023.0 2131.91  5029.5 2134.60  5035.3 2133.57
  5045.4 2137.48  5051.1 2137.02  5066.9 2152.06  5072.7 2151.81  5088.5 2162.46
  5094.3 2161.88  5110.1 2168.36  5126.0 2170.42  5131.7 2169.80  5189.0 2182.39
  5287.2 2193.15  5293.0 2192.55  5345.0 2199.35  5367.8 2201.60  5403.1 2201.94
#Mann=5,-1,0
  4600.0     0.1       0  4985.8    0.05       0  5009.3     0.1       0
  5189.0    0.07       0  5345.0     0.1       0
Bank Sta=4985.8,5009.3
Exp/Cntr=0.3,0.1

Type RM Length L Ch R = 1,16149,538,538,538
BEGIN DESCRIPTION:
Stream0095 28.0
END DESCRIPTION:
XS GIS Cut Line= 3
      1780025.02     13915825.01      1780375.00     13916075.00
      1780724.99     13916275.00
#Sta/Elev= 30
  4574.6 2167.66  4623.7 2163.44  4647.1 2162.58  4718.4 2155.73  4746.6 2154.58
  4789.6 2147.55  4819.1 2145.41  4881.8 2138.11  4918.7 2135.79  4932.2 2135.93
  4985.6 2131.25  4986.1 2130.75  5009.1 2131.25  5012.6 2136.07  5027.7 2139.59
  5034.2 2143.85  5040.0 2145.81  5062.3 2158.41  5077.4 2163.96  5093.2 2172.40
  5108.4 2177.30  5114.8 2180.71  5142.9 2187.12  5158.0 2189.53  5165.9 2191.92
  5195.5 2196.04  5232.9 2199.12  5319.3 2201.28  5356.7 2203.89  5407.8 2204.63
#Mann=3,-1,0
  4574.6     0.1       0  4985.6    0.05       0  5009.1     0.1       0
Bank Sta=4985.6,5009.1
Exp/Cntr=0.3,0.1

Type RM Length L Ch R = 1,15611,563,563,563
BEGIN DESCRIPTION:
Stream0095 27.0
END DESCRIPTION:
XS GIS Cut Line= 3
      1779774.98     13916324.99      1780125.00     13916525.00
      1780524.96     13916425.01
#Sta/Elev= 30
  4596.4 2167.11  4641.8 2164.50  4830.4 2149.03  4889.4 2142.13  4895.9 2138.97
  4905.2 2136.19  4926.8 2132.87  4979.9 2132.52  4980.4 2132.02  5003.4 2132.52
  5040.8 2133.58  5058.8 2137.50  5064.0 2136.66  5082.0 2138.86  5092.3 2140.60
  5100.0 2143.04  5105.2 2141.95  5112.9 2144.93  5141.3 2150.58  5146.4 2149.57
  5164.5 2154.42  5174.8 2156.14  5182.5 2158.72  5187.6 2157.87  5195.4 2160.93
  5246.9 2169.23  5265.0 2173.97  5298.3 2177.27  5370.6 2183.16  5411.8 2187.80
#Mann=4,-1,0
  4596.4     0.1       0  4979.9    0.05       0  5003.4     0.1       0
  5298.3   0.035       0
Bank Sta=4979.9,5003.4
Exp/Cntr=0.3,0.1

Type RM Length L Ch R = 1,15048,522,522,522
BEGIN DESCRIPTION:
Stream0095 26.0
END DESCRIPTION:
XS GIS Cut Line= 3
      1779525.03     13916675.03      1779825.00     13916975.00
      1780375.01     13916925.00
#Sta/Elev= 30
  4571.2 2171.02  4585.3 2171.06  4712.6 2164.72  4769.2 2162.99  4797.4 2161.15
  4811.6 2161.12  4894.7 2155.75  4910.6 2155.46  4938.9 2152.44  4953.0 2148.67
  4991.9 2133.64  4997.9 2133.64  5003.7 2131.38  5004.2 2130.88  5026.8 2130.88
  5027.3 2131.38  5045.1 2133.41  5055.7 2132.68  5065.7 2132.86  5075.8 2133.64
  5156.1 2135.74  5206.3 2134.83  5226.4 2137.03  5256.5 2142.22  5316.7 2150.41
  5367.0 2154.71  5394.4 2157.83  5427.2 2161.58  5487.4 2166.00  5547.7 2171.34
#Mann=6,-1,0
  4571.2   0.035       0  4894.7    0.07       0  5003.7    0.05       0
  5027.3    0.07       0  5045.1     0.1       0  5394.4   0.035       0
Bank Sta=5003.7,5027.3
Exp/Cntr=0.3,0.1

Type RM Length L Ch R = 1,14526,554,554,554
BEGIN DESCRIPTION:
Stream0095 25.0
END DESCRIPTION:
XS GIS Cut Line= 3
      1779625.03     13917724.97      1779925.00     13917425.00
      1780274.97     13917225.02
#Sta/Elev= 30
  4580.6 2188.73  4651.3 2187.47  4679.6 2184.35  4733.6 2180.83  4821.0 2174.02
  4835.1 2173.82  4849.3 2170.99  4877.5 2168.44  4905.8 2162.26  4920.0 2158.64
  4934.1 2144.87  4948.3 2135.53  4962.4 2130.01  4976.5 2127.41  4978.8 2125.26
  4979.3 2124.76  5002.0 2124.76  5002.5 2125.26  5004.8 2126.22  5027.9 2130.54
  5040.1 2131.83  5061.8 2132.72  5130.8 2135.25  5179.7 2139.47  5238.8 2148.02
  5271.9 2149.33  5350.3 2152.89  5378.4 2155.56  5394.3 2155.87  5407.9 2157.20
#Mann=6,-1,0
  4580.6     0.1       0  4733.6    0.07       0  4978.8    0.05       0
  5002.5    0.07       0  5061.8     0.1       0  5271.9   0.035       0
Bank Sta=4978.8,5002.5
Exp/Cntr=0.3,0.1

Type RM Length L Ch R = 1,13972,584,584,584
BEGIN DESCRIPTION:
Stream0095 24.0
END DESCRIPTION:
XS GIS Cut Line= 4
      1779925.04     13918024.98      1780275.00     13917825.00
      1780475.00     13917375.00      1780656.90     13916788.99
#Sta/Elev= 30
  4593.1 2181.59  4708.9 2175.61  4799.6 2173.36  4811.9 2170.93  4907.6 2164.97
  4929.2 2161.94  4945.1 2161.40  4950.8 2156.59  4960.9 2151.41  4966.7 2140.53
  4982.5 2135.59  4988.2 2128.42  4998.9 2127.61  5005.1 2124.98  5006.2 2122.89
  5006.7 2122.39  5029.9 2122.89  5050.9 2125.27  5072.8 2125.01  5116.5 2131.81
  5149.4 2133.85  5161.0 2136.05  5239.9 2140.06  5346.3 2145.11  5451.0 2155.47
  5491.2 2157.08  5645.7 2167.50  5802.7 2171.08  5959.8 2176.38  6102.2 2178.39
#Mann=5,-1,0
  4593.1     0.1       0  4960.9    0.07       0  5006.2    0.05       0
  5029.9    0.07       0  5239.9   0.035       0
Bank Sta=5006.2,5029.9
Exp/Cntr=0.3,0.1

Type RM Length L Ch R = 1,13388,1146,1146,1146
BEGIN DESCRIPTION:
Stream0095 23.0
END DESCRIPTION:
XS GIS Cut Line= 4
      1780475.04     13918124.98      1780825.00     13917925.00
      1781175.00     13917725.00      1781631.90     13917578.48
#Sta/Elev= 30
  4596.9 2159.73  4648.0 2158.98  4663.8 2156.48  4685.4 2155.05  4691.2 2155.79
  4750.2 2150.13  4861.8 2136.93  4896.3 2128.70  4927.3 2125.62  4942.4 2122.26
  4942.9 2121.76  4966.8 2122.26  4986.3 2124.27  4992.1 2123.28  4997.1 2124.14
  5045.3 2124.93  5072.7 2123.65  5088.5 2124.60  5110.1 2133.83  5115.9 2137.68
  5125.9 2140.70  5138.2 2148.81  5147.5 2151.19  5169.1 2153.87  5324.8 2159.64
  5419.1 2163.59  5476.6 2163.57  5665.6 2168.80  5783.0 2168.09  5882.9 2165.34
#Mann=4,-1,0
  4596.9     0.1       0  4942.4    0.05       0  4966.8     0.1       0
  5324.8    0.07       0
Bank Sta=4942.4,4966.8
Exp/Cntr=0.3,0.1

Type RM Length L Ch R = 1,12242,591,591,591
BEGIN DESCRIPTION:
Stream0095 22.0
END DESCRIPTION:
XS GIS Cut Line= 3
      1780675.01     13918225.01      1781475.00     13918725.00
      1781825.00     13918925.00
#Sta/Elev= 30
  4060.8 2149.47  4119.8 2146.83  4220.6 2137.83  4278.4 2135.89  4713.5 2133.91
  4750.1 2136.32  4756.5 2132.44  4765.4 2130.07  4771.3 2130.82  4780.1 2126.29
  4807.8 2129.83  4844.4 2129.09  4902.2 2124.27  4917.5 2120.52  4960.0 2117.78
  4968.9 2115.71  4969.4 2115.21  4993.5 2115.71  5001.2 2120.12  5007.1 2120.12
  5027.2 2128.75  5033.7 2139.60  5039.5 2137.09  5049.5 2142.79  5055.3 2142.72
  5061.8 2146.58  5071.1 2147.91  5173.4 2157.93  5269.1 2160.98  5407.3 2170.84
#Mann=3,-1,0
  4060.8     0.1       0  4968.9    0.05       0  4993.5     0.1       0
Bank Sta=4968.9,4993.5
Exp/Cntr=0.3,0.1

Type RM Length L Ch R = 1,11651,533,533,533
BEGIN DESCRIPTION:
Stream0095 21.0
END DESCRIPTION:
XS GIS Cut Line= 3
      1780324.97     13918374.97      1781125.00     13919175.00
      1781324.99     13919524.98
#Sta/Elev= 30
  3873.4 2166.50  4029.0 2154.57  4050.2 2151.84  4170.4 2143.97  4269.4 2138.56
  4396.7 2136.07  4495.7 2127.91  4566.4 2127.63  4665.4 2132.93  4722.0 2133.51
  4778.5 2132.12  4849.2 2127.52  4934.1 2118.32  4948.2 2115.61  4978.4 2113.31
  4978.9 2112.81  5003.0 2113.31  5004.8 2116.33  5018.5 2118.91  5027.8 2122.18
  5034.3 2127.48  5050.2 2136.76  5055.9 2138.44  5062.4 2143.76  5071.8 2149.14
  5077.5 2150.65  5211.4 2156.57  5217.2 2155.67  5319.4 2160.01  5407.9 2161.53
#Mann=3,-1,0
  3873.4     0.1       0  4978.4    0.05       0  5003.0     0.1       0
Bank Sta=4978.4,5003
Exp/Cntr=0.3,0.1

Type RM Length L Ch R = 1,11118,572,572,572
BEGIN DESCRIPTION:
Stream0095 20.0
END DESCRIPTION:
XS GIS Cut Line= 3
      1779924.97     13918624.97      1780675.00     13919425.00
      1781024.96     13919624.98
#Sta/Elev= 30
  3903.6 2174.77  4115.9 2156.78  4130.0 2154.71  4229.2 2148.42  4292.7 2140.86
  4363.5 2135.69  4427.0 2132.76  4568.7 2131.42  4639.5 2127.10  4802.2 2127.77
  4830.5 2125.32  4858.8 2120.15  4922.3 2118.58  4929.6 2117.10  5000.2 2113.61
  5001.6 2112.32  5002.1 2111.82  5026.3 2112.32  5035.5 2116.87  5057.8 2120.08
  5067.2 2122.63  5072.9 2126.11  5088.8 2128.43  5132.0 2139.79  5147.8 2141.39
  5153.6 2144.04  5169.4 2144.32  5175.2 2146.04  5228.4 2149.57  5403.3 2153.04
#Mann=3,-1,0
  3903.6     0.1       0  5001.6    0.05       0  5026.3     0.1       0
Bank Sta=5001.6,5026.3
Exp/Cntr=0.3,0.1

Type RM Length L Ch R = 1,10546,521,521,521
BEGIN DESCRIPTION:
Stream0095 19.0
END DESCRIPTION:
XS GIS Cut Line= 3
      1779925.01     13918825.03      1780175.00     13919625.00
      1780524.97     13919874.98
#Sta/Elev= 30
  4166.1 2158.43  4228.9 2153.23  4317.5 2148.94  4344.2 2146.52  4365.1 2143.92
  4382.4 2139.76  4387.7 2139.71  4414.9 2134.72  4511.8 2127.01  4742.3 2126.38
  4820.4 2121.75  4836.6 2118.68  4852.8 2117.55  4878.5 2117.84  4962.3 2113.96
  4999.2 2113.73  4999.7 2113.23  5023.9 2113.73  5026.3 2114.88  5041.1 2115.01
  5053.4 2118.21  5062.0 2118.91  5068.1 2122.11  5076.7 2123.93  5082.9 2126.77
  5118.5 2129.63  5148.0 2130.23  5248.8 2136.01  5376.6 2146.34  5434.3 2149.07
#Mann=3,-1,0
  4166.1     0.1       0  4999.2    0.05       0  5023.9     0.1       0
Bank Sta=4999.2,5023.9
Exp/Cntr=0.3,0.1

Type RM Length L Ch R = 1,10025,561,561,561
BEGIN DESCRIPTION:
Stream0095 18.0
END DESCRIPTION:
XS GIS Cut Line= 3
      1779324.96     13919825.00      1779725.00     13919825.00
      1780424.97     13919974.99
#Sta/Elev= 30
  4600.6 2172.45  4620.6 2171.52  4660.6 2171.27  4810.6 2164.52  4830.6 2162.81
  4850.6 2159.45  4860.6 2157.19  4900.6 2135.28  4910.6 2123.00  4920.6 2115.75
  4930.6 2111.33  4940.6 2109.25  4950.6 2109.59  4958.2 2108.61  4958.7 2108.11
  4983.0 2108.61  4998.1 2110.42  5051.8 2112.19  5092.7 2115.06  5154.0 2121.55
  5163.4 2123.18  5205.2 2125.87  5335.0 2129.95  5435.1 2130.57  5481.3 2130.53
  5548.6 2133.59  5573.4 2133.85  5598.1 2135.33  5691.8 2144.90  5716.5 2145.88
#Mann=5,-1,0
  4600.6     0.1       0  4958.2    0.05       0  4983.0     0.1       0
  5335.0    0.07       0  5435.1     0.1       0
Bank Sta=4958.2,4983
Exp/Cntr=0.3,0.1

Type RM Length L Ch R = 1,9464,548,548,548
BEGIN DESCRIPTION:
Stream0095 17.0
END DESCRIPTION:
XS GIS Cut Line= 3
      1779375.01     13920125.01      1779725.00     13920325.00
      1780446.67     13920026.94
#Sta/Elev= 30
  4592.4 2168.41  4826.3 2161.93  4857.3 2158.97  4863.8 2155.01  4869.5 2156.95
  4879.6 2149.62  4885.4 2155.85  4891.8 2141.36  4901.2 2135.74  4907.0 2137.66
  4914.9 2133.17  4922.8 2118.33  4928.6 2127.19  4937.9 2115.32  4944.4 2110.40
  4950.1 2113.66  4960.2 2104.13  4966.0 2107.27  4972.5 2103.04  4992.4 2100.95
  4992.9 2100.45  5017.2 2100.95  5034.1 2107.41  5058.0 2112.25  5111.2 2118.42
  5269.3 2124.15  5421.5 2124.27  5561.1 2129.26  5698.8 2143.06  5776.3 2146.01
#Mann=5,-1,0
  4592.4     0.1       0  4992.4    0.05       0  5017.2     0.1       0
  5269.3    0.07       0  5421.5     0.1       0
Bank Sta=4992.4,5017.2
Exp/Cntr=0.3,0.1

Type RM Length L Ch R = 1,8916,576,576,576
BEGIN DESCRIPTION:
Stream0095 16.0
END DESCRIPTION:
XS GIS Cut Line= 3
      1779674.99     13920775.00      1780075.00     13920725.00
      1780474.98     13920125.03
#Sta/Elev= 30
  4609.0 2158.48  4770.3 2152.72  4840.8 2148.87  4861.0 2146.44  4881.1 2142.75
  4888.7 2139.98  4893.7 2135.97  4901.3 2133.37  4921.4 2129.11  4931.5 2118.62
  4951.7 2108.36  4974.3 2103.28  4989.6 2102.43  4990.1 2101.93  5014.4 2102.43
  5019.6 2103.84  5048.2 2105.68  5061.7 2107.81  5112.8 2111.13  5133.8 2114.62
  5178.9 2116.85  5214.9 2120.16  5272.0 2121.99  5312.0 2121.65  5366.6 2121.50
  5431.3 2123.70  5488.4 2128.65  5560.5 2132.46  5611.5 2136.97  5733.2 2144.20
#Mann=5,-1,0
  4609.0     0.1       0  4989.6    0.05       0  5014.4     0.1       0
  5312.0    0.07       0  5366.6     0.1       0
Bank Sta=4989.6,5014.4
Exp/Cntr=0.3,0.1

Type RM Length L Ch R = 1,8340,583,583,583
BEGIN DESCRIPTION:
Stream0095 15.0
END DESCRIPTION:
XS GIS Cut Line= 3
      1780575.00     13921324.96      1780575.00     13920925.00
      1780731.74     13920123.34
#Sta/Elev= 30
  4595.8 2154.75  4625.8 2154.51  4675.8 2152.39  4845.8 2152.71  4915.8 2151.20
  4925.8 2149.49  4935.8 2143.95  4955.8 2131.62  4965.8 2120.86  4975.8 2111.71
  4985.8 2104.65  4993.3 2100.36  4998.3 2100.36  5003.7 2097.71  5004.2 2097.21
  5028.6 2097.71  5036.5 2100.57  5046.7 2101.09  5073.1 2105.65  5107.8 2108.62
  5124.6 2111.28  5335.8 2120.72  5398.1 2124.76  5454.3 2128.97  5464.5 2128.82
  5490.4 2130.75  5637.9 2137.27  5647.9 2138.09  5701.6 2139.27  5812.6 2144.36
#Mann=6,-1,0
  4595.8     0.1       0  5003.7    0.05       0  5028.6     0.1       0
  5398.1    0.07       0  5637.9     0.1       0  5647.9    0.07       0
Bank Sta=5003.7,5028.6
Exp/Cntr=0.3,0.1

Type RM Length L Ch R = 1,7757,528,528,528
BEGIN DESCRIPTION:
Stream0095 14.0
END DESCRIPTION:
XS GIS Cut Line= 3
      1780924.99     13921375.01      1781125.00     13921025.00
      1781329.97     13920019.82
#Sta/Elev= 30
  4592.9 2149.99  4718.9 2150.46  4821.1 2145.60  4848.5 2142.85  4864.3 2138.77
  4885.9 2136.73  4892.4 2133.20  4901.7 2130.49  4907.5 2130.54  4929.1 2126.30
  4938.4 2123.62  4944.9 2119.59  4950.7 2119.75  4966.5 2115.27  4982.4 2107.90
  4988.1 2108.15  4993.2 2104.40  4998.6 2104.40  5008.8 2098.82  5009.3 2098.32
  5033.7 2098.82  5098.1 2104.40  5172.9 2107.51  5218.4 2111.44  5414.5 2118.62
  5536.9 2128.99  5710.4 2133.10  5802.3 2137.53  5925.9 2141.01  6021.9 2146.48
#Mann=3,-1,0
  4592.9     0.1       0  5008.8    0.05       0  5033.7     0.1       0
Bank Sta=5008.8,5033.7
Exp/Cntr=0.3,0.1

Type RM Length L Ch R = 1,7229,556,556,556
BEGIN DESCRIPTION:
Stream0095 13.0
END DESCRIPTION:
XS GIS Cut Line= 3
      1781775.00     13921425.00      1781625.00     13921025.00
      1781637.45     13920003.38
#Sta/Elev= 30
  4568.0 2148.60  4583.1 2148.40  4685.5 2140.58  4803.0 2127.94  4814.5 2127.96
  4834.1 2125.44  4839.5 2125.96  4864.4 2122.10  4869.7 2122.42  4894.6 2115.21
  4900.0 2115.64  4919.6 2112.01  4924.9 2111.90  4949.8 2104.18  4955.2 2104.86
  4973.8 2102.66  4980.1 2103.52  4992.8 2102.19  4993.3 2101.69  5017.7 2102.19
  5135.2 2104.59  5285.2 2115.41  5295.2 2116.89  5425.2 2127.00  5485.2 2128.68
  5595.2 2127.93  5685.3 2128.81  5905.3 2137.60  5965.3 2141.93  6016.9 2142.65
#Mann=3,-1,0
  4568.0     0.1       0  4992.8    0.05       0  5017.7     0.1       0
Bank Sta=4992.8,5017.7
Exp/Cntr=0.3,0.1

Type RM Length L Ch R = 1,6673,600,600,600
BEGIN DESCRIPTION:
Stream0095 12.0
END DESCRIPTION:
XS GIS Cut Line= 3
      1782125.00     13921424.98      1782125.00     13921025.00
      1782275.00     13920225.02
#Sta/Elev= 30
  4595.6 2143.39  4645.6 2141.59  4665.6 2140.05  4775.6 2135.35  4805.6 2133.42
  4925.6 2116.49  4945.6 2112.17  4955.6 2108.58  4980.6 2102.42  4981.1 2101.92
  5005.1 2101.92  5005.6 2102.42  5138.0 2103.66  5148.2 2103.21  5199.1 2104.74
  5209.2 2104.30  5260.1 2107.00  5294.9 2107.33  5321.2 2108.49  5347.4 2107.96
  5382.2 2109.83  5443.2 2116.01  5473.8 2120.70  5562.8 2129.65  5567.9 2129.35
  5615.4 2134.73  5620.4 2134.75  5673.0 2143.99  5778.1 2153.45  5809.5 2155.56
#Mann=3,-1,0
  4595.6     0.1       0  4980.6    0.05       0  5005.6     0.1       0
Bank Sta=4980.6,5005.6
Exp/Cntr=0.3,0.1

Type RM Length L Ch R = 1,6073,378,378,378
BEGIN DESCRIPTION:
Stream0095 11.0
END DESCRIPTION:
XS GIS Cut Line= 3
      1782525.00     13921375.00      1782725.00     13921025.00
      1782425.00     13920225.01
#Sta/Elev= 30
  4596.9 2136.26  4648.0 2135.35  4744.5 2130.57  4919.4 2115.09  4942.4 2112.24
  4977.0 2106.04  4986.3 2102.12  4992.1 2101.97  4997.3 2098.49  4997.8 2097.99
  5022.3 2098.49  5075.7 2101.82  5130.8 2103.05  5149.5 2105.58  5186.0 2105.31
  5210.9 2106.94  5256.3 2105.96  5288.4 2102.99  5301.7 2103.27  5309.7 2101.65
  5341.8 2102.96  5395.2 2111.44  5467.3 2118.12  5512.7 2120.15  5630.1 2132.64
  5651.5 2133.95  5698.7 2139.70  5704.9 2141.79  5723.6 2143.98  5854.4 2154.59
#Mann=3,-1,0
  4596.9     0.1       0  4997.3    0.05       0  5022.3     0.1       0
Bank Sta=4997.3,5022.3
Exp/Cntr=0.3,0.1

Type RM Length L Ch R = 1,5695,758,758,758
BEGIN DESCRIPTION:
Stream0095 10.0
END DESCRIPTION:
XS GIS Cut Line= 3
      1783075.00     13921324.98      1783089.11     13920900.54
      1784038.13     13919459.78
#Sta/Elev= 30
  4649.8 2123.15  4749.8 2119.63  4889.9 2109.41  4919.9 2105.81  4959.9 2098.40
  4997.5 2095.40  4998.0 2094.90  5022.5 2095.40  5050.0 2097.95  5069.7 2102.66
  5090.7 2105.69  5132.8 2107.82  5205.1 2106.28  5298.4 2097.76  5313.5 2099.26
  5356.5 2108.58  5400.9 2111.59  5560.1 2115.34  5638.8 2119.30  5732.1 2121.71
  5768.3 2123.30  5783.3 2125.23  5883.4 2129.33  5955.2 2134.70  6051.0 2136.27
  6129.7 2139.66  6244.1 2147.80  6403.7 2155.46  6584.4 2160.15  6799.7 2168.15
#Mann=3,-1,0
  4649.8     0.1       0  4997.5    0.05       0  5022.5     0.1       0
Bank Sta=4997.5,5022.5
Exp/Cntr=0.3,0.1

Type RM Length L Ch R = 1,4937,539,539,539
BEGIN DESCRIPTION:
Stream0095 9.0
END DESCRIPTION:
XS GIS Cut Line= 3
      1783124.96     13921375.02      1783775.00     13921075.00
      1784124.96     13920875.02
#Sta/Elev= 30
  4283.8 2123.68  4338.5 2121.61  4487.1 2111.78  4601.9 2108.67  4735.4 2106.92
  4834.5 2100.63  4870.8 2096.26  4900.6 2094.49  4955.7 2092.97  4968.1 2094.08
  4994.9 2092.79  4995.4 2092.29  5020.4 2092.79  5022.8 2094.48  5028.5 2095.85
  5035.0 2104.17  5057.3 2113.04  5066.7 2114.85  5080.4 2119.49  5103.4 2121.16
  5153.1 2128.38  5168.9 2129.69  5174.7 2131.28  5190.5 2132.04  5212.1 2135.71
  5227.9 2135.89  5287.0 2140.71  5308.5 2143.54  5330.1 2144.21  5402.8 2150.67
#Mann=3,-1,0
  4283.8     0.1       0  4994.9    0.05       0  5020.4     0.1       0
Bank Sta=4994.9,5020.4
Exp/Cntr=0.3,0.1

Type RM Length L Ch R = 1,4398,575,575,575
BEGIN DESCRIPTION:
Stream0095 8.0
END DESCRIPTION:
XS GIS Cut Line= 3
      1783225.01     13921475.00      1783925.00     13921525.00
      1784275.01     13921725.01
#Sta/Elev= 30
  4298.3 2120.10  4348.4 2118.65  4366.0 2116.80  4528.9 2108.68  4709.3 2105.90
  4869.7 2101.01  4932.4 2096.93  4990.0 2088.87  5000.1 2088.90  5000.9 2086.89
  5001.4 2086.39  5026.6 2086.89  5029.6 2088.37  5035.3 2088.09  5051.2 2090.94
  5057.7 2093.90  5067.0 2107.82  5072.8 2110.19  5080.7 2121.07  5088.6 2129.65
  5094.4 2131.57  5103.7 2138.44  5110.2 2140.77  5131.8 2140.71  5175.0 2145.03
  5265.0 2151.71  5271.5 2153.49  5307.8 2155.69  5389.5 2158.68  5403.2 2160.26
#Mann=4,-1,0
  4298.3     0.1       0  5000.9    0.05       0  5026.6     0.1       0
  5307.8    0.07       0
Bank Sta=5000.9,5026.6
Exp/Cntr=0.3,0.1

Type RM Length L Ch R = 1,3823,566,566,566
BEGIN DESCRIPTION:
Stream0095 7.0
END DESCRIPTION:
XS GIS Cut Line= 3
      1783275.01     13921725.01      1783725.00     13922025.00
      1784074.97     13922224.98
#Sta/Elev= 30
  4454.8 2114.62  4519.4 2111.36  4534.4 2111.35  4555.4 2109.44  4663.6 2104.51
  4771.8 2100.99  4837.9 2099.80  4864.9 2097.61  4901.0 2096.19  4937.0 2092.26
  4952.1 2089.24  4979.8 2086.33  4980.3 2085.83  5005.5 2086.33  5030.9 2090.12
  5041.0 2090.78  5053.2 2095.93  5068.3 2113.20  5076.2 2124.30  5082.0 2129.67
  5084.2 2135.05  5089.9 2138.82  5099.3 2141.57  5121.6 2144.35  5143.2 2148.64
  5164.8 2149.96  5192.1 2153.93  5208.0 2154.35  5233.5 2157.36  5398.7 2164.60
#Mann=4,-1,0
  4454.8     0.1       0  4979.8    0.05       0  5005.5     0.1       0
  5233.5    0.07       0
Bank Sta=4979.8,5005.5
Exp/Cntr=0.3,0.1

Type RM Length L Ch R = 1,3257,513,513,513
BEGIN DESCRIPTION:
Stream0095 6.0
END DESCRIPTION:
XS GIS Cut Line= 3
      1782625.03     13922325.00      1783425.00     13922475.00
      1783824.98     13922574.99
#Sta/Elev= 30
  4186.1 2141.44  4236.9 2138.14  4328.5 2128.95  4501.5 2118.76  4562.5 2113.04
  4595.6 2108.96  4623.6 2103.07  4633.7 2101.99  4648.2 2098.05  4684.6 2096.67
  4725.3 2097.40  4786.4 2096.13  4827.1 2093.93  4863.5 2090.59  4908.4 2090.19
  4949.1 2087.97  4979.7 2089.57  4984.6 2086.53  4985.1 2086.03  5010.3 2086.53
  5018.1 2086.65  5059.3 2092.50  5092.8 2102.48  5146.9 2115.07  5175.2 2122.91
  5206.2 2132.65  5237.1 2144.20  5278.3 2155.10  5389.1 2168.07  5412.3 2169.65
#Mann=3,-1,0
  4186.1     0.1       0  4984.6    0.05       0  5010.3     0.1       0
Bank Sta=4984.6,5010.3
Exp/Cntr=0.3,0.1

Type RM Length L Ch R = 1,2744,553,553,553
BEGIN DESCRIPTION:
Stream0095 5.0
END DESCRIPTION:
XS GIS Cut Line= 3
      1782475.02     13922325.01      1783225.00     13922925.00
      1783625.04     13922975.01
#Sta/Elev= 30
  4044.1 2152.28  4094.5 2150.07  4144.1 2144.46  4214.6 2141.32  4307.4 2130.55
  4449.9 2122.06  4534.7 2114.22  4598.7 2105.18  4620.4 2094.67  4627.6 2092.92
  4648.4 2090.40  4656.4 2091.40  4685.1 2087.03  4685.6 2086.53  4710.9 2087.03
  4712.4 2089.39  4798.8 2091.57  4976.5 2089.68  5034.8 2092.91  5065.0 2098.43
  5145.6 2100.31  5165.8 2103.32  5208.6 2114.36  5236.3 2125.14  5266.6 2132.56
  5284.2 2140.79  5289.2 2140.41  5306.9 2146.08  5364.8 2153.81  5407.7 2156.75
#Mann=3,-1,0
  4044.1     0.1       0  4685.1    0.05       0  4710.9     0.1       0
Bank Sta=4685.1,4710.9
Exp/Cntr=0.3,0.1

Type RM Length L Ch R = 1,2191,511,511,511
BEGIN DESCRIPTION:
Stream0095 4.0
END DESCRIPTION:
XS GIS Cut Line= 3
      1782675.01     13922875.02      1782875.00     13923225.00
      1783339.40     13923391.71
#Sta/Elev= 30
  4592.8 2117.21  4696.4 2110.94  4724.5 2110.43  4789.3 2105.94  4799.4 2106.16
  4869.9 2100.29  4907.3 2095.86  4944.8 2093.45  4966.4 2090.15  4982.2 2089.30
  4993.0 2085.80  4998.5 2085.80  5004.2 2081.42  5004.7 2080.92  5030.0 2081.42
  5036.7 2083.36  5049.0 2084.94  5067.4 2086.11  5091.5 2085.33  5144.6 2087.40
  5240.3 2097.11  5277.2 2105.43  5282.8 2107.95  5293.4 2109.96  5314.6 2116.92
  5333.4 2121.18  5369.5 2132.48  5389.0 2136.85  5400.2 2141.20  5489.3 2149.05
#Mann=3,-1,0
  4592.8     0.1       0  5004.2    0.05       0  5030.0     0.1       0
Bank Sta=5004.2,5030
Exp/Cntr=0.3,0.1

Type RM Length L Ch R = 1,1680,516,516,516
BEGIN DESCRIPTION:
Stream0095 3.0
END DESCRIPTION:
XS GIS Cut Line= 3
      1782374.99     13923274.99      1782775.00     13923675.00
      1783174.99     13923625.00
#Sta/Elev= 30
  4434.3 2112.48  4462.6 2111.81  4519.2 2107.98  4604.0 2104.35  4703.0 2095.68
  4745.4 2093.66  4802.0 2088.50  4830.3 2088.32  4858.6 2086.73  4872.7 2084.74
  4886.9 2085.98  4915.1 2082.70  4929.3 2082.63  4957.6 2080.10  4971.7 2081.53
  4985.9 2081.68  4997.2 2080.07  4997.7 2079.57  5023.0 2080.07  5037.8 2085.67
  5042.8 2083.21  5070.5 2094.47  5090.7 2106.35  5110.9 2114.71  5118.4 2119.28
  5123.4 2115.37  5141.1 2124.99  5181.4 2141.93  5352.7 2148.75  5403.1 2149.46
#Mann=3,-1,0
  4434.3     0.1       0  4997.2    0.05       0  5023.0     0.1       0
Bank Sta=4997.2,5023
Exp/Cntr=0.3,0.1

Type RM Length L Ch R = 1,1164,559,559,559
BEGIN DESCRIPTION:
Stream0095 2.0
END DESCRIPTION:
XS GIS Cut Line= 3
      1782174.99     13923474.99      1782375.00     13923825.00
      1782325.01     13924224.96
#Sta/Elev= 30
  4589.1 2106.77  4646.7 2104.76  4656.1 2103.49  4661.8 2103.95  4779.9 2096.47
  4903.7 2091.20  4934.6 2087.56  4941.1 2085.81  4969.2 2084.61  4978.6 2081.73
  4984.3 2081.16  4989.4 2075.79  4989.9 2075.29  5015.3 2075.79  5022.5 2077.12
  5042.6 2078.01  5082.9 2077.62  5093.0 2079.62  5103.1 2082.84  5110.6 2088.27
  5115.7 2088.42  5123.2 2097.91  5136.9 2108.45  5153.5 2120.74  5163.6 2130.97
  5173.6 2139.24  5183.7 2141.30  5203.9 2142.77  5294.6 2144.36  5395.3 2144.29
#Mann=4,-1,0
  4589.1     0.1       0  4989.4    0.05       0  5015.3     0.1       0
  5136.9    0.07       0
Bank Sta=4989.4,5015.3
Exp/Cntr=0.3,0.1

Type RM Length L Ch R = 1,605,325,325,325
BEGIN DESCRIPTION:
Stream0095 1.0
END DESCRIPTION:
XS GIS Cut Line= 3
      1781925.00     13923625.00      1781875.00     13924025.00
      1782224.98     13924224.99
#Sta/Elev= 30
  4601.8 2100.20  4672.3 2096.26  4692.5 2096.98  4783.2 2092.69  4805.9 2090.99
  4843.7 2084.49  4886.5 2081.73  4904.1 2078.10  4984.8 2075.71  4999.9 2073.16
  5000.4 2072.66  5025.8 2073.16  5028.0 2076.20  5034.4 2077.43  5040.2 2081.49
  5050.3 2085.44  5056.0 2094.70  5071.9 2096.80  5077.6 2100.39  5085.5 2101.09
  5093.5 2103.92  5108.6 2109.43  5120.8 2116.24  5130.9 2118.83  5143.1 2125.91
  5152.5 2127.26  5195.7 2139.49  5313.7 2145.34  5372.4 2145.91  5408.0 2146.17
#Mann=4,-1,0
  4601.8     0.1       0  4999.9    0.05       0  5025.8     0.1       0
  5372.4    0.07       0
Bank Sta=4999.9,5025.8
Exp/Cntr=0.3,0.1

Type RM Length L Ch R = 1,280,0,0,0
BEGIN DESCRIPTION:
Stream0095 0.0
END DESCRIPTION:
XS GIS Cut Line= 4
      1781599.86     13923153.52      1781512.52     13923922.94
      1781656.09     13924312.10      1781910.92     13924472.39
#Sta/Elev= 30
  4065.8 2113.07  4228.3 2107.04  4242.6 2105.71  4349.1 2103.04  4429.6 2102.46
  4610.8 2097.45  4775.3 2089.17  4822.1 2088.01  4865.4 2084.43  4885.0 2080.37
  4890.5 2077.72  4963.5 2071.97  4964.0 2071.47  4989.4 2071.97  5023.6 2072.76
  5067.8 2077.33  5087.5 2081.20  5098.2 2086.47  5118.0 2091.16  5123.3 2093.37
  5162.1 2101.76  5172.8 2103.11  5215.4 2114.35  5257.3 2122.36  5277.3 2127.23
  5285.9 2127.61  5343.6 2135.91  5395.4 2140.92  5466.3 2145.34  5556.0 2145.10
#Mann=3,-1,0
  4065.8     0.1       0  4963.5    0.05       0  4989.4     0.1       0
Bank Sta=4963.5,4989.4
Exp/Cntr=0.3,0.1

Chan Stop Cuts=-1
