--- West Dry Branch.prj (project) ---

Proj Title=West Dry Branch Base Level Engineering
Current Plan=p01
Default Exp/Contr=0.3,0.1
English Units
Geom File=g01
Flow File=f01
Plan File=p01
BEGIN DESCRIPTION:
West Dry Branch
END DESCRIPTION:

--- West Dry Branch.p01 (plan) ---

Plan Title=Multiple Run
Short Identifier=Multiple
Geom File=g01
Flow File=f01
Subcritical Flow
K Sum by GR= 0
Std Step Tol= 0.01
Critical Tol= 0.01
Num of Std Step Trials= 20
Max Error Tol= 0.3
Flow Tol Ratio= 0.001
Split Flow NTrial= 30
Split Flow Tol= 0.02
Split Flow Ratio= 0.02
Log Output Level= 0
Friction Slope Method= 1
Unsteady Friction Slope Method= 2
Unsteady Bridges Friction Slope Method= 1
Parabolic Critical Depth
Global Vel Dist=  1 , 1 , 1
Global Log Level= 0
CheckData=True
Encroach Param= -1, 0, 0, 0
BEGIN DESCRIPTION:
Multiple Run
END DESCRIPTION:

--- West Dry Branch.f01 (steady flow) ---

Flow Title=Multiple
Number of Profiles=7
Profile Names=10-year,25-year,50-year,1pct_min,100-year,1pct_plu,500-year
River Rch & RM= West Dry Branch,Reach-1,31899
     539     880    1190     780    1557    3107    2628
River Rch & RM= West Dry Branch,Reach-1,30231
    1265    2159    3010    2025    4040    8061    7195
River Rch & RM= West Dry Branch,Reach-1,22817
    2574    4552    6494    4460    8899   17755   16530
River Rch & RM= West Dry Branch,Reach-1,16504
    3009    5354    7671    5288   10551   21052   19749
River Rch & RM= West Dry Branch,Reach-1,6341
    3313    5920    8503    5875   11722   23389   22041
Boundary for River Rch & Prof#=West Dry Branch,Reach-1,1
Up Type=0
Dn Type=3
Dn Slope=0.005
Boundary for River Rch & Prof#=West Dry Branch,Reach-1,2
Up Type=0
Dn Type=3
Dn Slope=0.005
Boundary for River Rch & Prof#=West Dry Branch,Reach-1,3
Up Type=0
Dn Type=3
Dn Slope=0.005
Boundary for River Rch & Prof#=West Dry Branch,Reach-1,4
Up Type=0
Dn Type=3
Dn Slope=0.005
Boundary for River Rch & Prof#=West Dry Branch,Reach-1,5
Up Type=0
Dn Type=3
Dn Slope=0.005
Boundary for River Rch & Prof#=West Dry Branch,Reach-1,6
Up Type=0
Dn Type=3
Dn Slope=0.005
Boundary for River Rch & Prof#=West Dry Branch,Reach-1,7
Up Type=0
Dn Type=3
Dn Slope=0.005

--- West Dry Branch.g01 (geometry) ---

Geom Title=Existing Conditions

River Reach=West Dry Branch,Reach-1
Reach XY= 30
      1868275.00     13990025.00      1867325.38     13986940.16
      1867523.96     13986664.35      1867478.76     13986026.56
      1868222.73     13985119.06      1868284.41     13983818.38
      1868515.29     13983435.75      1869122.94     13983169.15
      1868932.56     13982025.00      1869224.62     13981240.16
      1868227.06     13979969.14      1868471.39     13978426.50
      1867577.14     13977719.03      1867921.25     13976576.55
      1866774.51     13975540.20      1866782.81     13975268.81
      1867773.78     13974114.50      1867771.55     13973676.25
      1867228.45     13972876.49      1868038.35     13972461.64
      1868174.63     13972040.27      1867388.62     13971388.24
      1867041.68     13970691.64      1866097.72     13970149.14
      1865774.70     13969595.18      1866211.47     13968988.55
      1866919.92     13968669.96      1867433.30     13967578.06
      1868914.52     13967573.81      1869325.00     13967225.00

Type RM Length L Ch R = 1,31899,455,455,455
BEGIN DESCRIPTION:
West Dry Branch 69.0
END DESCRIPTION:
XS GIS Cut Line= 3
      1868475.02     13990025.01      1868325.00     13989925.00
      1868074.96     13989975.01
#Sta/Elev= 30
  4819.8 2164.41  4842.4 2163.36  4848.4 2163.55  4891.9 2161.20  4914.5 2161.05
  4920.5 2160.39  4928.0 2160.64  4935.5 2160.08  4950.5 2159.78  4964.0 2158.38
  4971.6 2156.84  4977.6 2156.40  4986.6 2154.19  4992.6 2154.00  4995.1 2153.44
  4995.3 2152.94  4998.8 2152.94  4999.1 2153.44  5002.7 2153.44  5010.3 2155.34
  5020.5 2156.27  5030.7 2156.08  5061.3 2157.53  5071.5 2157.44  5091.9 2159.39
  5122.5 2160.75  5163.3 2163.44  5193.9 2164.95  5234.7 2168.29  5255.1 2169.14
#Mann=3,-1,0
  4819.8    0.07       0  4995.1    0.05       0  4999.1    0.07       0
Bank Sta=4995.1,4999.1
Exp/Cntr=0.3,0.1

Type RM Length L Ch R = 1,31444,421,421,421
BEGIN DESCRIPTION:
West Dry Branch 68.0
END DESCRIPTION:
XS GIS Cut Line= 3
      1868324.96     13989475.01      1868175.00     13989525.00
      1868074.97     13989675.04
#Sta/Elev= 30
  4841.7 2157.57  4852.2 2157.28  4873.3 2156.07  4883.8 2155.30  4894.4 2154.19
  4904.9 2153.64  4936.5 2150.18  4947.1 2149.31  4968.1 2146.62  4987.2 2145.27
  4987.5 2144.77  4991.0 2144.77  4991.2 2145.27  4997.1 2145.90  5002.8 2145.90
  5007.3 2146.79  5013.3 2146.81  5022.3 2147.26  5028.3 2147.22  5043.3 2148.26
  5071.9 2150.70  5079.4 2151.75  5085.4 2151.95  5094.4 2152.72  5121.5 2156.13
  5130.5 2156.69  5144.0 2158.21  5151.5 2158.22  5166.5 2159.02  5180.1 2159.32
#Mann=3,-1,0
  4841.7    0.07       0  4987.2    0.05       0  4991.2    0.07       0
Bank Sta=4987.2,4991.2
Exp/Cntr=0.3,0.1

Type RM Length L Ch R = 1,31023,471,471,471
BEGIN DESCRIPTION:
West Dry Branch 67.0
END DESCRIPTION:
XS GIS Cut Line= 3
      1868125.02     13989175.00      1867975.00     13989175.00
      1867824.98     13989425.03
#Sta/Elev= 30
  4850.0 2149.26  4880.0 2148.01  4900.0 2146.71  4940.0 2142.99  4950.0 2142.50
  4960.0 2140.94  4970.0 2140.24  4980.0 2139.21  4995.5 2138.78  4995.8 2138.28
  4999.3 2138.28  4999.5 2138.78  5002.9 2138.78  5035.0 2140.47  5044.7 2140.75
  5050.6 2140.55  5066.1 2141.33  5071.9 2140.57  5081.7 2140.24  5093.3 2140.69
  5103.0 2141.38  5108.9 2142.75  5124.4 2143.70  5130.2 2144.31  5140.0 2144.68
  5167.2 2147.17  5198.3 2149.13  5225.5 2151.56  5278.0 2154.25  5291.6 2154.69
#Mann=3,-1,0
  4850.0    0.07       0  4995.5    0.05       0  4999.5    0.07       0
Bank Sta=4995.5,4999.5
Exp/Cntr=0.3,0.1

Type RM Length L Ch R = 1,30552,321,321,321
BEGIN DESCRIPTION:
West Dry Branch 66.0
END DESCRIPTION:
XS GIS Cut Line= 3
      1867974.97     13988824.99      1867775.00     13988775.00
      1867675.03     13988824.99
#Sta/Elev= 30
  4799.8 2139.90  4817.8 2139.62  4851.3 2137.89  4859.0 2137.20  4864.2 2137.25
  4882.2 2136.68  4900.3 2135.22  4905.4 2135.41  4933.8 2133.75  4941.5 2132.99
  4946.7 2133.29  4964.7 2130.33  4982.7 2128.76  4987.9 2129.41  4993.5 2128.38
  4993.6 2128.36  4993.9 2127.86  4997.4 2127.86  4997.6 2128.36  5003.4 2129.54
  5008.7 2129.54  5014.3 2131.70  5019.9 2132.61  5028.3 2134.99  5036.7 2136.14
  5050.6 2137.47  5059.0 2138.01  5064.6 2138.03  5081.4 2139.18  5117.7 2141.05
#Mann=4,-1,0
  4799.8     0.1       0  4993.5    0.07       0  4993.6    0.05       0
  4997.6    0.07       0
Bank Sta=4993.6,4997.6
Exp/Cntr=0.3,0.1

Type RM Length L Ch R = 1,30231,438,438,438
BEGIN DESCRIPTION:
West Dry Branch 65.0
END DESCRIPTION:
XS GIS Cut Line= 3
      1867975.02     13988374.99      1867693.51     13988482.58
      1867575.04     13988524.99
#Sta/Elev= 30
  4691.2 2142.17  4706.3 2142.40  4723.3 2140.37  4755.5 2138.83  4761.0 2136.97
  4766.4 2137.54  4785.7 2134.08  4791.1 2134.35  4798.3 2132.83  4815.8 2131.08
  4821.2 2131.72  4835.4 2130.68  4862.5 2128.81  4870.6 2128.43  4875.9 2128.85
  4894.6 2127.87  4898.6 2127.11  4898.9 2126.61  4902.4 2126.61  4902.6 2127.11
  4906.0 2128.09  4910.8 2127.79  4960.8 2127.83  4980.1 2128.45  5022.9 2127.76
  5033.5 2129.17  5041.5 2131.23  5065.3 2135.64  5072.3 2136.36  5118.4 2137.65
#Mann=5,-1,0
  4691.2   0.035       0  4835.4    0.07       0  4898.6   0.035       0
  4902.6    0.07       0  4910.8   0.035       0
Bank Sta=4898.6,4902.6
Exp/Cntr=0.3,0.1

Type RM Length L Ch R = 1,29793,179,179,179
BEGIN DESCRIPTION:
West Dry Branch 4.1
END DESCRIPTION:
XS GIS Cut Line= 3
      1867930.16     13987860.55      1867757.43     13988069.49
      1867509.47     13988299.50
#Sta/Elev= 30
  4684.9 2143.84  4748.5 2141.33  4791.5 2140.67  4805.8 2139.97  4812.3 2138.88
  4820.2 2139.10  4826.6 2137.51  4841.0 2137.89  4847.5 2136.61  4884.0 2133.50
  4890.5 2131.93  4904.8 2131.09  4911.3 2129.25  4919.1 2128.72  4940.0 2121.44
  4954.0 2119.77  4961.4 2120.26  4966.8 2119.65  4967.0 2119.15  4970.8 2119.65
  4989.8 2119.89  4997.1 2121.08  5039.6 2121.54  5074.8 2123.00  5082.1 2122.36
  5131.5 2123.81  5138.3 2123.36  5145.7 2124.25  5174.0 2124.52  5294.2 2128.46
#Mann=3,-1,0
  4684.9   0.035       0  4966.8   0.035       0  4970.8   0.035       0
Bank Sta=4966.8,4970.8
Exp/Cntr=0.3,0.1

Type RM Length L Ch R = 1,29614,447,447,447
BEGIN DESCRIPTION:
West Dry Branch 64.0
END DESCRIPTION:
XS GIS Cut Line= 3
      1867828.45     13987748.99      1867625.00     13987975.00
      1867324.96     13988175.03
#Sta/Elev= 30
  4700.7 2138.76  4742.8 2137.05  4799.6 2129.96  4853.6 2126.25  4863.2 2124.86
  4877.4 2125.42  4884.1 2123.87  4891.6 2124.21  4898.3 2122.54  4905.8 2122.64
  4912.5 2120.76  4926.7 2119.61  4981.5 2117.39  4981.7 2116.89  4985.5 2117.39
  5001.4 2118.86  5018.3 2117.94  5033.3 2119.42  5063.4 2119.17  5105.5 2120.75
  5120.5 2119.88  5126.5 2120.66  5135.5 2119.52  5141.5 2120.73  5149.0 2120.06
  5171.6 2123.33  5213.6 2124.71  5239.1 2126.90  5300.8 2131.84  5365.4 2134.59
#Mann=6,-1,0
  4700.7   0.035       0  4799.6     0.1       0  4853.6   0.035       0
  4981.5   0.035       0  4985.5   0.035       0  5239.1    0.07       0
Bank Sta=4981.5,4985.5
Exp/Cntr=0.3,0.1

Type RM Length L Ch R = 1,29167,453,453,453
BEGIN DESCRIPTION:
West Dry Branch 63.0
END DESCRIPTION:
XS GIS Cut Line= 3
      1867725.01     13987625.00      1867425.00     13987625.00
      1867125.03     13987724.99
#Sta/Elev= 30
  4699.4 2129.94  4701.9 2129.94  4709.4 2128.50  4759.4 2122.93  4790.9 2118.79
  4819.4 2116.28  4899.4 2114.48  4949.4 2114.58  4959.4 2114.17  4969.4 2112.86
  4979.4 2113.06  4987.4 2112.57  4987.7 2112.07  4991.2 2112.07  4991.4 2112.57
  4996.9 2114.16  5020.5 2114.82  5031.0 2114.70  5041.6 2116.00  5083.7 2116.72
  5115.4 2118.62  5125.9 2120.34  5147.0 2120.98  5168.1 2122.78  5199.7 2123.15
  5252.4 2125.13  5273.5 2126.15  5284.0 2127.57  5305.1 2128.24  5315.6 2129.15
#Mann=4,-1,0
  4699.4     0.1       0  4790.9    0.07       0  4987.4    0.05       0
  4991.4    0.07       0
Bank Sta=4987.4,4991.4
Exp/Cntr=0.3,0.1

Type RM Length L Ch R = 1,28714,456,456,456
BEGIN DESCRIPTION:
West Dry Branch 62.0
END DESCRIPTION:
XS GIS Cut Line= 3
      1867790.89     13987238.77      1867375.00     13987225.00
      1867174.98     13987275.01
#Sta/Elev= 30
  4588.7 2123.14  4594.6 2122.46  4603.0 2122.39  4704.7 2115.75  4734.7 2115.12
  4754.7 2115.36  4764.7 2114.41  4804.7 2112.79  4851.7 2111.56  4874.8 2111.38
  4914.8 2109.90  4964.8 2109.64  4975.9 2108.58  4992.8 2105.48  4993.1 2104.98
  4996.6 2104.98  4996.8 2105.48  5002.3 2107.32  5015.1 2106.79  5022.9 2108.42
  5028.0 2108.69  5035.7 2108.47  5076.9 2109.20  5097.6 2108.82  5128.5 2109.62
  5151.7 2112.08  5169.7 2115.10  5180.1 2117.39  5200.7 2119.12  5211.0 2119.25
#Mann=6,-1,0
  4588.7   0.035       0  4603.0    0.07       0  4975.9   0.035       0
  4992.8   0.035       0  4996.8   0.035       0  5076.9    0.07       0
Bank Sta=4992.8,4996.8
Exp/Cntr=0.3,0.1

Type RM Length L Ch R = 1,28258,442,442,442
BEGIN DESCRIPTION:
West Dry Branch 61.0
END DESCRIPTION:
XS GIS Cut Line= 3
      1867674.98     13987024.98      1867425.00     13986825.00
      1867124.97     13986774.99
#Sta/Elev= 30
  4680.1 2112.78  4708.1 2112.70  4722.5 2111.54  4772.1 2109.29  4815.3 2108.00
  4821.7 2108.62  4829.7 2107.58  4879.4 2106.14  4943.4 2105.40  4957.8 2104.56
  4978.6 2104.08  4993.0 2102.25  5010.4 2102.37  5018.5 2101.60  5018.8 2101.10
  5022.3 2101.10  5022.5 2101.60  5033.2 2104.01  5050.9 2104.56  5088.9 2105.03
  5154.8 2104.96  5210.6 2106.73  5215.7 2106.55  5233.4 2107.44  5263.8 2111.44
  5271.4 2113.39  5276.5 2113.43  5284.1 2115.95  5301.8 2120.33  5304.4 2120.33
#Mann=3,-1,0
  4680.1    0.07       0  5018.5    0.05       0  5022.5    0.07       0
Bank Sta=5018.5,5022.5
Exp/Cntr=0.3,0.1

Type RM Length L Ch R = 1,27816,463,463,463
BEGIN DESCRIPTION:
West Dry Branch 60.0
END DESCRIPTION:
XS GIS Cut Line= 3
      1867674.98     13986624.99      1867425.00     13986475.00
      1867124.96     13986575.01
#Sta/Elev= 30
  4708.0 2105.69  4801.3 2103.67  4847.9 2103.62  4869.3 2102.74  4875.1 2103.24
  4890.7 2101.96  4896.5 2103.21  4906.2 2101.84  4912.1 2099.90  4917.9 2100.34
  4927.6 2097.21  4933.4 2098.39  4941.2 2096.86  4949.0 2097.04  4954.8 2096.28
  4983.9 2094.92  4984.2 2094.42  4987.7 2094.42  4987.9 2094.92  5002.2 2095.48
  5010.1 2098.13  5031.2 2100.22  5136.6 2101.66  5178.7 2103.00  5210.3 2105.23
  5242.0 2109.53  5284.1 2113.24  5305.2 2115.97  5313.1 2117.98  5315.8 2117.98
#Mann=3,-1,0
  4708.0    0.07       0  4983.9    0.05       0  4987.9    0.07       0
Bank Sta=4983.9,4987.9
Exp/Cntr=0.3,0.1

Type RM Length L Ch R = 1,27353,443,443,443
BEGIN DESCRIPTION:
West Dry Branch 59.0
END DESCRIPTION:
XS GIS Cut Line= 3
      1867725.02     13986325.02      1867475.00     13986025.00
      1867424.97     13985974.97
#Sta/Elev= 30
  4614.2 2101.85  4656.5 2100.82  4685.2 2099.06  4692.3 2098.98  4699.5 2098.00
  4734.6 2096.25  4777.6 2095.03  4820.6 2093.25  4862.2 2093.40  4898.7 2092.63
  4919.5 2093.60  4933.8 2093.23  4940.3 2092.30  4948.1 2092.09  4954.6 2092.50
  4968.9 2092.56  4976.8 2091.98  4983.3 2090.25  4989.1 2089.46  4989.3 2088.96
  4992.8 2088.96  4993.1 2089.46  4997.6 2090.29  5001.5 2089.78  5008.3 2089.78
  5018.9 2092.02  5033.0 2098.93  5040.1 2099.88  5047.2 2102.00  5075.5 2103.18
#Mann=3,-1,0
  4614.2    0.07       0  4989.1    0.05       0  4993.1    0.07       0
Bank Sta=4989.1,4993.1
Exp/Cntr=0.3,0.1

Type RM Length L Ch R = 1,26910,420,420,420
BEGIN DESCRIPTION:
West Dry Branch 58.0
END DESCRIPTION:
XS GIS Cut Line= 3
      1868075.04     13985925.03      1867775.00     13985725.00
      1867625.01     13985675.00
#Sta/Elev= 30
  4635.1 2102.08  4657.7 2101.74  4663.7 2101.35  4671.2 2101.48  4695.4 2099.87
  4699.7 2099.88  4707.3 2096.51  4720.8 2095.55  4743.3 2095.18  4756.8 2094.25
  4765.8 2092.46  4792.9 2089.64  4807.9 2089.19  4859.0 2088.89  4901.1 2088.07
  4960.5 2088.25  4986.2 2086.20  4986.4 2085.70  4989.9 2085.70  4990.2 2086.20
  4992.7 2086.66  5006.2 2086.63  5027.3 2087.42  5037.9 2088.81  5048.4 2091.07
  5101.1 2095.54  5111.7 2096.94  5132.7 2097.50  5143.3 2098.53  5153.8 2099.04
#Mann=5,-1,0
  4635.1    0.07       0  4695.4   0.035       0  4960.5    0.07       0
  4986.2    0.05       0  4990.2    0.07       0
Bank Sta=4986.2,4990.2
Exp/Cntr=0.3,0.1

Type RM Length L Ch R = 1,26490,476,476,476
BEGIN DESCRIPTION:
West Dry Branch 57.0
END DESCRIPTION:
XS GIS Cut Line= 3
      1868225.01     13985575.01      1868025.00     13985425.00
      1867724.95     13985374.99
#Sta/Elev= 30
  4750.2 2101.89  4778.3 2099.93  4792.9 2098.30  4813.8 2094.49  4828.3 2090.96
  4842.9 2090.66  4857.5 2086.20  4872.1 2084.00  4892.9 2082.97  4913.8 2082.82
  4972.1 2083.74  4978.3 2083.40  4984.2 2081.02  4986.7 2080.01  4990.9 2079.44
  4991.2 2078.94  4994.7 2078.94  4994.9 2079.44  4997.1 2081.33  5002.7 2081.33
  5010.4 2084.93  5020.5 2086.96  5050.9 2086.77  5061.0 2085.52  5071.2 2086.09
  5088.9 2088.36  5154.8 2089.72  5220.1 2093.49  5243.5 2095.08  5304.4 2097.83
#Mann=5,-1,0
  4750.2    0.07       0  4984.2   0.035       0  4990.9   0.035       0
  4994.9   0.035       0  5220.1    0.07       0
Bank Sta=4990.9,4994.9
Exp/Cntr=0.3,0.1

Type RM Length L Ch R = 1,26014,444,444,444
BEGIN DESCRIPTION:
West Dry Branch 56.0
END DESCRIPTION:
XS GIS Cut Line= 3
      1868425.03     13985075.01      1868225.00     13985025.00
      1867975.03     13985074.99
#Sta/Elev= 30
  4793.5 2097.32  4803.8 2097.19  4811.6 2095.54  4824.5 2094.71  4845.1 2092.68
  4852.8 2090.96  4858.0 2090.54  4865.7 2088.55  4887.4 2085.67  4899.2 2083.88
  4906.9 2081.74  4935.3 2077.87  4940.4 2077.56  4968.8 2078.48  4976.5 2079.09
  4989.4 2078.94  4997.1 2076.67  5007.9 2076.32  5008.1 2075.82  5011.6 2075.82
  5011.9 2076.32  5081.3 2082.17  5091.5 2082.39  5111.9 2083.77  5177.8 2085.81
  5203.6 2086.55  5213.8 2086.45  5224.0 2087.50  5234.2 2087.90  5254.6 2087.45
#Mann=5,-1,0
  4793.5     0.1       0  4887.4    0.07       0  5007.9    0.05       0
  5011.9    0.07       0  5177.8   0.035       0
Bank Sta=5007.9,5011.9
Exp/Cntr=0.3,0.1

Type RM Length L Ch R = 1,25570,480,480,480
BEGIN DESCRIPTION:
West Dry Branch 55.0
END DESCRIPTION:
XS GIS Cut Line= 3
      1868524.99     13984724.99      1868275.00     13984625.00
      1868124.96     13984675.01
#Sta/Elev= 30
  4730.6 2092.23  4752.1 2091.66  4769.6 2090.27  4775.0 2090.49  4823.5 2084.72
  4828.9 2084.64  4846.6 2082.95  4870.6 2080.37  4877.3 2078.58  4882.7 2078.40
  4892.1 2076.07  4901.6 2074.80  4906.9 2074.40  4924.5 2075.18  4936.6 2075.26
  4960.8 2074.02  4985.0 2072.02  4988.4 2071.42  4988.7 2070.92  4992.2 2070.92
  4992.4 2071.42  5002.5 2071.69  5010.4 2072.93  5020.9 2073.79  5031.5 2075.93
  5042.0 2077.48  5052.5 2078.34  5136.9 2080.74  5147.4 2081.79  5158.0 2081.51
#Mann=4,-1,0
  4730.6     0.1       0  4846.6    0.07       0  4988.4    0.05       0
  4992.4    0.07       0
Bank Sta=4988.4,4992.4
Exp/Cntr=0.3,0.1

Type RM Length L Ch R = 1,25090,451,451,451
BEGIN DESCRIPTION:
West Dry Branch 54.0
END DESCRIPTION:
XS GIS Cut Line= 3
      1868574.98     13984474.98      1868275.00     13984175.00
      1867974.98     13984225.00
#Sta/Elev= 30
  4580.3 2085.33  4622.7 2084.47  4693.4 2081.51  4721.7 2079.63  4778.3 2077.07
  4800.3 2075.14  4849.0 2070.90  4872.3 2071.42  4905.5 2071.32  4933.8 2071.76
  4948.0 2071.33  4969.2 2069.97  4974.3 2068.62  4974.5 2068.12  4978.0 2068.12
  4978.3 2068.62  4990.4 2068.66  5001.0 2069.75  5007.1 2069.75  5024.8 2071.19
  5032.4 2071.40  5045.1 2072.70  5085.6 2074.37  5136.3 2075.67  5146.5 2076.48
  5217.1 2077.46  5227.6 2078.21  5268.1 2079.57  5288.4 2080.83  5308.7 2081.20
#Mann=6,-1,0
  4580.3     0.1       0  4800.3    0.07       0  4872.3     0.1       0
  4974.3    0.05       0  4978.3     0.1       0  5217.1   0.035       0
Bank Sta=4974.3,4978.3
Exp/Cntr=0.3,0.1

Type RM Length L Ch R = 1,24639,423,423,423
BEGIN DESCRIPTION:
West Dry Branch 53.0
END DESCRIPTION:
XS GIS Cut Line= 3
      1868724.97     13984074.98      1868325.00     13983775.00
      1868174.98     13983574.97
#Sta/Elev= 30
  4494.3 2081.16  4501.6 2081.44  4507.8 2080.57  4622.4 2078.17  4766.1 2074.06
  4822.4 2069.14  4830.7 2067.66  4857.8 2066.16  4900.5 2066.82  4922.4 2068.17
  4937.0 2066.67  4951.6 2068.09  4972.4 2067.28  4987.0 2066.14  4989.0 2065.27
  4989.3 2064.77  4993.0 2064.77  4993.2 2065.27  5001.6 2065.65  5007.8 2066.86
  5051.6 2066.78  5080.7 2067.63  5087.0 2069.48  5101.6 2071.74  5107.8 2074.56
  5122.4 2076.43  5151.6 2079.32  5180.7 2081.07  5207.8 2084.87  5244.3 2088.38
#Mann=3,-1,0
  4494.3     0.1       0  4989.0    0.05       0  4993.2     0.1       0
Bank Sta=4989,4993.2
Exp/Cntr=0.3,0.1

Type RM Length L Ch R = 1,24216,914,914,914
BEGIN DESCRIPTION:
West Dry Branch 52.0
END DESCRIPTION:
XS GIS Cut Line= 3
      1868924.98     13983824.98      1868525.00     13983425.00
      1868375.03     13983325.02
#Sta/Elev= 30
  4439.1 2083.84  4467.4 2082.40  4495.6 2078.52  4538.1 2074.74  4580.5 2072.19
  4778.5 2065.66  4820.9 2065.33  4849.2 2064.09  4877.5 2064.27  4905.8 2062.99
  4948.2 2063.82  4962.3 2062.04  4990.6 2061.77  5001.2 2064.24  5012.3 2064.28
  5027.3 2064.02  5033.3 2063.02  5048.3 2063.38  5052.2 2061.66  5052.5 2061.16
  5056.4 2061.66  5063.4 2061.81  5069.4 2064.39  5084.4 2065.27  5099.4 2067.95
  5105.4 2069.90  5112.9 2070.39  5122.9 2072.64  5162.5 2081.99  5185.0 2083.74
#Mann=4,-1,0
  4439.1     0.1       0  5052.2    0.05       0  5056.4     0.1       0
  5122.9   0.035       0
Bank Sta=5052.2,5056.4
Exp/Cntr=0.3,0.1

Type RM Length L Ch R = 1,23302,485,485,485
BEGIN DESCRIPTION:
West Dry Branch 51.0
END DESCRIPTION:
XS GIS Cut Line= 3
      1869224.98     13982975.00      1869125.00     13982975.00
      1868325.00     13983175.00
#Sta/Elev= 30
  4900.4 2069.28  4920.4 2069.52  4960.4 2066.97  4980.4 2062.67  4990.4 2058.75
  4997.9 2052.82  5003.0 2052.82  5008.5 2050.17  5008.8 2049.67  5012.8 2050.17
  5018.4 2052.88  5031.3 2054.41  5041.6 2054.32  5072.5 2056.60  5082.8 2056.73
  5106.0 2055.26  5113.8 2056.34  5175.6 2057.23  5216.8 2059.43  5250.1 2059.67
  5353.4 2063.11  5412.7 2066.06  5567.3 2070.45  5645.1 2071.57  5683.3 2073.52
  5732.2 2078.64  5752.8 2080.03  5765.7 2082.25  5788.9 2083.03  5825.0 2085.16
#Mann=6,-1,0
  4900.4     0.1       0  5008.5    0.05       0  5012.8     0.1       0
  5250.1    0.07       0  5645.1     0.1       0  5788.9    0.07       0
Bank Sta=5008.5,5012.8
Exp/Cntr=0.3,0.1

Type RM Length L Ch R = 1,22817,455,455,455
BEGIN DESCRIPTION:
West Dry Branch 50.0
END DESCRIPTION:
XS GIS Cut Line= 3
      1869424.96     13982475.01      1869125.00     13982525.00
      1868725.01     13982724.99
#Sta/Elev= 30
  4695.9 2065.87  4728.8 2064.75  4746.6 2062.48  4777.0 2061.37  4833.7 2057.73
  4888.5 2054.37  4898.6 2052.94  4915.3 2051.87  4972.1 2051.52  4989.9 2049.88
  4994.1 2048.61  4994.6 2048.11  5000.3 2048.11  5000.8 2048.61  5002.8 2048.61
  5008.4 2051.09  5014.0 2052.37  5053.1 2052.66  5081.1 2050.18  5103.4 2050.03
  5134.2 2051.00  5142.5 2052.03  5156.5 2051.07  5164.9 2051.20  5192.9 2052.14
  5232.0 2055.20  5246.0 2055.28  5290.7 2058.39  5343.8 2060.90  5447.2 2064.04
#Mann=5,-1,0
  4695.9    0.07       0  4833.7     0.1       0  4915.3    0.07       0
  4994.1    0.05       0  5000.8    0.07       0
Bank Sta=4994.1,5000.8
Exp/Cntr=0.3,0.1

Type RM Length L Ch R = 1,22362,447,447,447
BEGIN DESCRIPTION:
West Dry Branch 49.0
END DESCRIPTION:
XS GIS Cut Line= 3
      1869374.96     13982274.98      1868975.00     13982125.00
      1868825.03     13982224.98
#Sta/Elev= 30
  4572.8 2062.51  4618.1 2060.42  4627.0 2059.46  4753.4 2052.63  4758.8 2053.17
  4771.9 2052.17  4813.9 2052.38  4829.1 2051.30  4874.5 2050.01  4899.4 2049.99
  4924.3 2048.38  4959.9 2047.46  4978.6 2048.05  4990.2 2047.46  4997.3 2045.86
  5003.0 2045.86  5010.1 2044.77  5010.6 2044.27  5016.4 2044.27  5016.9 2044.77
  5028.5 2045.21  5043.5 2047.13  5049.5 2047.08  5058.5 2050.36  5064.6 2050.35
  5079.6 2053.93  5100.6 2055.29  5125.8 2058.60  5171.5 2060.76  5180.2 2061.41
#Mann=7,-1,0
  4572.8   0.035       0  4627.0     0.1       0  4771.9   0.035       0
  5010.1   0.035       0  5016.9   0.035       0  5125.8    0.07       0
  5171.5   0.035       0
Bank Sta=5010.1,5016.9
Exp/Cntr=0.3,0.1

Type RM Length L Ch R = 1,21915,476,476,476
BEGIN DESCRIPTION:
West Dry Branch 48.0
END DESCRIPTION:
XS GIS Cut Line= 3
      1869425.03     13982125.03      1869025.00     13981725.00
      1868824.99     13981775.00
#Sta/Elev= 30
  4433.8 2061.49  4448.0 2061.34  4565.7 2055.39  4592.6 2053.74  4617.7 2052.70
  4700.8 2051.19  4716.7 2050.12  4751.4 2049.25  4826.7 2048.26  4900.5 2046.66
  4937.6 2045.02  4941.9 2044.73  4967.5 2043.62  4968.0 2043.12  4974.4 2043.12
  4974.9 2043.62  5002.1 2045.05  5009.8 2045.99  5040.8 2045.71  5053.6 2044.47
  5064.0 2044.53  5071.7 2045.30  5082.0 2047.18  5100.0 2052.32  5105.2 2052.26
  5112.9 2054.10  5141.3 2057.46  5146.4 2056.91  5174.8 2058.54  5205.7 2058.97
#Mann=11,-1,0
  4433.8   0.035       0  4565.7    0.07       0  4592.6     0.1       0
  4700.8    0.07       0  4751.4     0.1       0  4826.7    0.07       0
  4937.6     0.1       0  4941.9    0.07       0  4967.5    0.05       0
  4974.9    0.07       0  5053.6     0.1       0
Bank Sta=4967.5,4974.9
Exp/Cntr=0.3,0.1

Type RM Length L Ch R = 1,21439,362,362,362
BEGIN DESCRIPTION:
West Dry Branch 47.0
END DESCRIPTION:
XS GIS Cut Line= 3
      1869525.04     13981224.99      1869225.00     13981325.00
      1868775.00     13981625.00
#Sta/Elev= 30
  4683.9 2081.24  4726.1 2076.80  4768.3 2070.16  4821.0 2064.50  4852.6 2060.52
  4863.1 2059.98  4921.1 2050.90  4989.6 2042.69  4993.8 2040.13  4994.3 2039.63
  5000.8 2039.63  5001.3 2040.13  5013.7 2040.32  5043.7 2042.73  5049.7 2042.33
  5058.8 2043.47  5072.3 2043.10  5130.9 2044.76  5136.9 2044.43  5157.9 2045.13
  5230.0 2045.93  5281.1 2044.61  5288.6 2043.12  5302.1 2041.60  5311.1 2043.95
  5315.7 2044.31  5324.7 2046.80  5368.2 2050.63  5446.4 2054.56  5541.0 2056.26
#Mann=3,-1,0
  4683.9    0.07       0  4993.8    0.05       0  5001.3    0.07       0
Bank Sta=4993.8,5001.3
Exp/Cntr=0.3,0.1

Type RM Length L Ch R = 1,21077,185,185,185
BEGIN DESCRIPTION:
West Dry Branch 46.0
END DESCRIPTION:
XS GIS Cut Line= 3
      1869380.01     13981012.57      1869081.65     13981021.47
      1868378.72     13981036.95
#Sta/Elev= 30
  4688.7 2071.01  4707.2 2070.17  4723.7 2069.55  4793.8 2063.43  4808.9 2060.34
  4833.8 2057.37  4922.6 2049.30  4943.8 2047.07  5033.9 2040.37  5053.9 2039.36
  5073.9 2039.94  5083.9 2039.30  5103.9 2039.51  5120.1 2038.45  5120.6 2037.95
  5127.1 2037.95  5127.6 2038.45  5143.9 2040.21  5153.9 2040.14  5173.9 2043.09
  5183.9 2042.86  5193.9 2041.64  5213.9 2041.22  5243.9 2043.34  5263.9 2042.78
  5343.9 2043.93  5383.9 2046.82  5454.0 2047.98  5604.0 2052.32  5690.3 2052.84
#Mann=6,-1,0
  4688.7    0.07       0  4707.2     0.1       0  4808.9    0.07       0
  4922.6   0.035       0  5120.1   0.035       0  5127.6   0.035       0
Bank Sta=5120.1,5127.6
Exp/Cntr=0.3,0.1

Type RM Length L Ch R = 1,20892,389,389,389
BEGIN DESCRIPTION:
West Dry Branch 45.2
END DESCRIPTION:
XS GIS Cut Line= 2
      1869347.27     13980955.18      1868393.61     13980929.54
#Sta/Elev= 30
  4576.7 2068.90  4629.0 2066.17  4659.0 2062.67  4669.0 2061.24  4704.8 2053.64
  4729.0 2048.38  4766.7 2043.33  4771.8 2044.12  4789.0 2042.06  4829.1 2040.07
  4859.1 2040.73  4889.1 2040.30  4919.1 2039.10  4939.1 2036.47  4979.1 2036.38
  4985.3 2035.48  4985.8 2034.98  4992.4 2034.98  4992.9 2035.48  5029.1 2037.16
  5069.1 2042.12  5137.8 2042.11  5142.9 2041.69  5199.2 2042.26  5269.2 2044.97
  5299.2 2044.87  5329.2 2045.57  5379.3 2047.82  5469.3 2049.62  5530.7 2049.69
#Mann=4,-1,0
  4576.7     0.1       0  4704.8    0.07       0  4985.3    0.05       0
  4992.9    0.07       0
Bank Sta=4985.3,4992.9
Exp/Cntr=0.3,0.1

Type RM Length L Ch R = 1,20503,450,450,450
BEGIN DESCRIPTION:
West Dry Branch 45.0
END DESCRIPTION:
XS GIS Cut Line= 3
      1869074.99     13980625.00      1868725.00     13980625.00
      1868325.00     13980675.00
#Sta/Elev= 30
  4650.5 2053.77  4670.5 2053.37  4700.5 2050.99  4750.5 2049.01  4770.5 2046.99
  4800.5 2044.92  4860.5 2042.20  4890.5 2039.54  4900.5 2039.31  4910.5 2038.02
  4920.5 2035.82  4930.5 2035.06  4950.5 2035.31  4970.5 2034.48  4980.5 2033.44
  5020.6 2036.27  5038.3 2035.33  5050.9 2035.40  5071.0 2033.71  5101.3 2033.21
  5115.0 2032.31  5115.5 2031.81  5122.4 2031.81  5122.9 2032.31  5141.6 2034.88
  5181.9 2036.78  5199.5 2039.33  5232.3 2041.86  5302.8 2045.08  5403.6 2052.14
#Mann=3,-1,0
  4650.5    0.07       0  5115.0    0.05       0  5122.9    0.07       0
Bank Sta=5115,5122.9
Exp/Cntr=0.3,0.1

Type RM Length L Ch R = 1,20053,438,438,438
BEGIN DESCRIPTION:
West Dry Branch 44.0
END DESCRIPTION:
XS GIS Cut Line= 3
      1868825.01     13980275.00      1868425.00     13980375.00
      1868055.49     13980593.11
#Sta/Elev= 30
  4595.8 2048.28  4655.1 2045.13  4688.6 2044.79  4791.7 2039.85  4832.9 2037.47
  4853.5 2034.71  4884.4 2032.72  4907.6 2033.32  4925.7 2031.46  4936.0 2032.48
  4948.9 2035.77  4956.6 2036.53  4966.9 2035.25  4977.2 2032.10  4984.9 2031.71
  4986.1 2031.01  4986.6 2030.51  4994.1 2031.01  5011.0 2031.83  5015.9 2033.25
  5021.7 2032.60  5031.3 2034.22  5058.8 2034.39  5074.5 2038.97  5160.7 2046.60
  5218.8 2051.44  5262.7 2053.84  5277.4 2054.48  5394.2 2059.53  5437.2 2061.13
#Mann=7,-1,0
  4595.8    0.07       0  4986.1    0.05       0  4994.1    0.07       0
  5160.7   0.035       0  5262.7    0.07       0  5277.4   0.035       0
  5394.2    0.07       0
Bank Sta=4986.1,4994.1
Exp/Cntr=0.3,0.1

Type RM Length L Ch R = 1,19615,450,450,450
BEGIN DESCRIPTION:
West Dry Branch 43.0
END DESCRIPTION:
XS GIS Cut Line= 3
      1869074.99     13979775.00      1868275.00     13980025.00
      1867869.58     13980038.97
#Sta/Elev= 30
  4161.8 2065.17  4298.0 2056.70  4307.9 2055.44  4345.7 2053.00  4410.6 2049.97
  4415.9 2050.54  4423.7 2049.57  4465.6 2047.84  4551.0 2046.06  4610.7 2043.06
  4633.2 2043.06  4790.4 2035.45  4848.5 2033.62  4905.6 2033.11  4926.6 2032.02
  4978.5 2031.76  5005.8 2030.82  5006.3 2030.32  5014.0 2030.82  5030.0 2033.68
  5050.0 2039.47  5145.1 2050.14  5160.0 2049.90  5190.1 2052.72  5259.7 2056.47
  5280.1 2057.64  5300.1 2057.79  5320.1 2059.20  5350.1 2059.11  5405.6 2061.65
#Mann=4,-1,0
  4161.8    0.07       0  5005.8    0.05       0  5014.0    0.07       0
  5259.7   0.035       0
Bank Sta=5005.8,5014
Exp/Cntr=0.3,0.1

Type RM Length L Ch R = 1,19165,422,422,422
BEGIN DESCRIPTION:
West Dry Branch 42.0
END DESCRIPTION:
XS GIS Cut Line= 3
      1868906.55     13979636.71      1868325.00     13979625.00
      1868174.97     13979625.00
#Sta/Elev= 30
  4413.8 2053.87  4525.4 2049.21  4545.4 2049.06  4575.4 2047.87  4585.4 2047.15
  4645.4 2045.42  4715.4 2041.30  4725.4 2041.18  4735.4 2040.08  4795.4 2036.79
  4805.4 2035.85  4835.4 2034.00  4875.4 2032.17  4915.5 2031.00  4965.5 2031.83
  4975.5 2031.01  4985.5 2028.28  4993.0 2024.22  5001.3 2024.09  5001.8 2023.59
  5009.1 2023.59  5009.6 2024.09  5015.5 2024.50  5045.5 2024.33  5055.5 2025.76
  5075.5 2031.84  5095.5 2039.09  5105.5 2041.70  5143.0 2047.72  5145.5 2047.72
#Mann=3,-1,0
  4413.8    0.07       0  5001.3    0.05       0  5009.6    0.07       0
Bank Sta=5001.3,5009.6
Exp/Cntr=0.3,0.1

Type RM Length L Ch R = 1,18743,425,425,425
BEGIN DESCRIPTION:
West Dry Branch 41.0
END DESCRIPTION:
XS GIS Cut Line= 3
      1868846.78     13979112.69      1868421.33     13979230.19
      1868059.89     13979406.90
#Sta/Elev= 30
  4551.2 2050.63  4652.7 2041.53  4800.4 2031.19  4840.0 2031.04  4853.9 2029.66
  4874.3 2030.32  4879.5 2028.76  4913.9 2026.81  5017.7 2024.24  5018.2 2023.74
  5026.1 2024.24  5032.6 2025.64  5038.1 2025.04  5055.1 2032.35  5060.6 2030.44
  5066.4 2034.06  5083.2 2037.15  5088.7 2035.47  5105.7 2037.59  5111.2 2035.29
  5128.2 2038.32  5133.8 2036.73  5150.7 2038.77  5156.3 2038.03  5173.2 2039.88
  5218.3 2041.75  5223.8 2040.97  5240.8 2042.87  5268.9 2043.20  5394.9 2050.22
#Mann=3,-1,0
  4551.2   0.035       0  5017.7   0.035       0  5026.1   0.035       0
Bank Sta=5017.7,5026.1
Exp/Cntr=0.3,0.1

Type RM Length L Ch R = 1,18318,92,92,92
BEGIN DESCRIPTION:
West Dry Branch 40.1
END DESCRIPTION:
XS GIS Cut Line= 3
      1868852.98     13978752.80      1868432.00     13978835.21
      1867970.84     13978932.60
#Sta/Elev= 30
  4614.5 2050.49  4706.6 2045.08  4744.9 2040.24  4758.1 2039.99  4785.7 2036.87
  4804.5 2035.76  4809.6 2036.77  4827.4 2035.34  4867.2 2035.27  4907.5 2033.74
  4912.6 2035.51  4928.3 2034.03  4938.5 2031.60  4958.9 2024.53  4964.1 2021.50
  4995.4 2021.02  4995.9 2020.52  5004.0 2021.02  5026.3 2024.00  5053.1 2026.28
  5066.3 2027.92  5071.4 2030.36  5101.7 2029.45  5116.0 2030.75  5127.7 2030.37
  5255.0 2032.64  5418.6 2039.06  5439.0 2040.69  5449.0 2040.19  5514.8 2042.72
#Mann=7,-1,0
  4614.5   0.035       0  4827.4   0.063       0  4995.4    0.05       0
  5004.0   0.063       0  5026.3    0.07       0  5053.1   0.063       0
  5127.7   0.035       0
Bank Sta=4995.4,5004
Exp/Cntr=0.3,0.1

Type RM Length L Ch R = 1,18226,172,172,172
BEGIN DESCRIPTION:
West Dry Branch 40.0
END DESCRIPTION:
XS GIS Cut Line= 3
      1868954.05     13978736.63      1868507.90     13978744.77
      1868010.98     13978752.66
#Sta/Elev= 30
  4551.0 2052.99  4580.1 2053.86  4602.4 2053.02  4700.1 2047.76  4735.5 2045.06
  4740.5 2045.11  4800.1 2038.86  4850.1 2035.69  4910.1 2033.76  4950.1 2033.25
  4960.1 2032.16  4991.9 2019.69  4992.4 2019.19  5000.0 2019.19  5000.5 2019.69
  5020.1 2020.31  5030.1 2021.85  5052.7 2023.62  5060.1 2023.80  5080.1 2026.38
  5100.1 2027.50  5180.1 2029.05  5250.2 2031.19  5290.2 2032.93  5325.9 2035.12
  5330.9 2033.34  5348.7 2034.51  5400.2 2037.76  5489.7 2045.80  5494.2 2045.80
#Mann=6,-1,0
  4551.0   0.063       0  4602.4   0.035       0  4991.9   0.035       0
  5000.5   0.035       0  5052.7    0.07       0  5348.7   0.035       0
Bank Sta=4991.9,5000.5
Exp/Cntr=0.3,0.1

Type RM Length L Ch R = 1,18054,706,706,706
BEGIN DESCRIPTION:
West Dry Branch 39.0
END DESCRIPTION:
XS GIS Cut Line= 3
      1868902.75     13978589.40      1868528.13     13978601.80
      1867878.37     13978644.78
#Sta/Elev= 30
  4622.3 2049.05  4637.8 2047.57  4642.8 2047.92  4780.1 2038.28  4850.2 2033.92
  4900.2 2031.83  4938.9 2029.32  4943.9 2029.77  4970.2 2022.56  4980.2 2021.20
  5001.2 2020.28  5016.0 2018.53  5016.5 2018.03  5024.1 2018.03  5024.6 2018.53
  5040.3 2020.04  5050.4 2022.27  5060.4 2021.58  5080.4 2025.07  5090.5 2025.03
  5123.4 2026.36  5160.6 2025.90  5260.8 2027.15  5274.3 2027.94  5351.0 2028.69
  5420.2 2030.25  5425.3 2030.76  5531.4 2032.52  5576.2 2034.25  5648.3 2037.93
#Mann=3,-1,0
  4622.3    0.07       0  5016.0    0.05       0  5024.6    0.07       0
Bank Sta=5016,5024.6
Exp/Cntr=0.3,0.1

Type RM Length L Ch R = 1,17348,186,186,186
BEGIN DESCRIPTION:
West Dry Branch 38.0
END DESCRIPTION:
XS GIS Cut Line= 3
      1868225.03     13978074.99      1868075.00     13978125.00
      1867725.02     13978474.98
#Sta/Elev= 30
  4836.8 2031.73  4889.5 2028.22  4910.6 2027.46  4942.2 2022.48  4952.8 2018.96
  4973.9 2016.41  4980.0 2013.95  4980.5 2013.45  4988.3 2013.45  4988.8 2013.95
  5009.1 2014.20  5023.2 2017.85  5065.7 2018.68  5079.8 2019.49  5122.2 2020.73
  5150.5 2021.23  5178.8 2021.03  5263.6 2023.19  5277.8 2024.04  5298.1 2024.58
  5320.2 2025.16  5348.5 2026.61  5376.8 2027.28  5390.9 2028.88  5405.1 2031.13
  5419.2 2034.38  5461.6 2042.64  5475.8 2043.52  5486.4 2044.95  5489.9 2044.95
#Mann=4,-1,0
  4836.8    0.07       0  4980.0    0.05       0  4988.8    0.07       0
  5298.1   0.035       0
Bank Sta=4980,4988.8
Exp/Cntr=0.3,0.1

Type RM Length L Ch R = 1,17162,207,207,207
BEGIN DESCRIPTION:
West Dry Branch 37.1
END DESCRIPTION:
XS GIS Cut Line= 3
      1868128.43     13977660.69      1867880.34     13978104.28
      1867759.18     13978314.16
#Sta/Elev= 30
  4578.7 2030.95  4606.6 2030.77  4620.1 2028.04  4636.1 2030.46  4673.2 2029.89
  4776.5 2027.55  4857.6 2024.13  4928.4 2018.24  4966.1 2017.18  4983.3 2014.52
  4983.8 2014.02  4992.4 2014.52  5025.5 2015.66  5047.2 2014.99  5106.4 2019.58
  5149.5 2024.68  5186.8 2026.65  5192.6 2027.79  5224.1 2027.61  5229.9 2028.50
  5245.7 2027.75  5251.4 2029.10  5267.2 2028.33  5273.0 2030.19  5283.0 2029.71
  5288.8 2032.16  5304.5 2031.76  5310.3 2034.50  5326.1 2034.44  5329.3 2036.61
#Mann=4,-1,0
  4578.7   0.094       0  4673.2   0.035       0  4983.3   0.035       0
  4992.4   0.035       0
Bank Sta=4983.3,4992.4
Exp/Cntr=0.3,0.1

Type RM Length L Ch R = 1,16955,451,451,451
BEGIN DESCRIPTION:
West Dry Branch 37.0
END DESCRIPTION:
XS GIS Cut Line= 3
      1867991.52     13977601.10      1867743.52     13977950.12
      1867639.31     13978118.40
#Sta/Elev= 30
  4576.5 2026.98  4627.6 2025.65  4669.4 2025.46  4678.0 2025.04  4684.1 2022.83
  4691.7 2021.58  4713.7 2020.91  4745.1 2021.10  4850.2 2018.52  4877.2 2016.07
  4885.9 2016.39  4892.0 2015.53  4942.4 2017.03  4978.1 2016.23  4992.9 2012.11
  4999.0 2011.37  5000.0 2010.68  5000.5 2010.18  5008.6 2010.18  5009.1 2010.68
  5022.2 2011.24  5035.1 2014.42  5044.6 2017.79  5050.4 2021.40  5057.5 2023.96
  5071.7 2027.84  5081.0 2029.14  5151.5 2033.34  5187.5 2034.33  5202.6 2035.93
#Mann=4,-1,0
  4576.5   0.094       0  4745.1   0.035       0  5000.0   0.035       0
  5009.1   0.035       0
Bank Sta=5000,5009.1
Exp/Cntr=0.3,0.1

Type RM Length L Ch R = 1,16504,485,485,485
BEGIN DESCRIPTION:
West Dry Branch 36.0
END DESCRIPTION:
XS GIS Cut Line= 3
      1867975.03     13977575.00      1867625.00     13977575.00
      1867525.03     13977575.00
#Sta/Elev= 30
  4645.4 2027.57  4685.4 2027.56  4695.4 2026.17  4705.4 2023.22  4720.9 2021.73
  4735.4 2020.05  4755.4 2019.11  4805.4 2018.01  4815.4 2018.28  4845.4 2016.91
  4850.1 2016.34  4865.4 2014.84  4875.4 2014.79  4885.4 2015.29  4915.4 2015.30
  4945.4 2016.15  4965.4 2014.75  4975.4 2012.62  4985.4 2011.34  5010.8 2009.95
  5011.3 2009.45  5019.6 2009.45  5020.1 2009.95  5025.4 2010.44  5035.4 2010.21
  5045.4 2012.62  5055.4 2019.98  5065.4 2026.09  5075.4 2029.12  5095.4 2030.25
#Mann=5,-1,0
  4645.4   0.094       0  4720.9     0.1       0  4850.1    0.07       0
  5010.8    0.05       0  5020.1    0.07       0
Bank Sta=5010.8,5020.1
Exp/Cntr=0.3,0.1

Type RM Length L Ch R = 1,16019,476,476,476
BEGIN DESCRIPTION:
West Dry Branch 35.0
END DESCRIPTION:
XS GIS Cut Line= 3
      1868025.03     13977125.00      1867725.00     13977125.00
      1867524.99     13977175.00
#Sta/Elev= 30
  4699.5 2024.25  4739.5 2023.00  4781.2 2020.69  4809.5 2019.22  4819.5 2020.00
  4839.5 2014.19  4859.5 2011.70  4899.8 2009.71  4919.5 2009.56  4929.5 2008.32
  4949.5 2008.45  4964.8 2006.75  4965.3 2006.25  4974.2 2006.75  4979.5 2006.82
  4997.0 2009.62  5009.8 2009.51  5022.7 2007.56  5040.8 2008.76  5051.1 2009.67
  5058.8 2011.62  5064.0 2012.14  5071.7 2014.90  5092.3 2016.78  5100.0 2018.44
  5112.9 2019.85  5146.4 2021.26  5154.1 2022.83  5164.5 2022.55  5205.7 2024.96
#Mann=5,-1,0
  4699.5    0.07       0  4781.2     0.1       0  4899.8    0.07       0
  4964.8    0.05       0  4974.2    0.07       0
Bank Sta=4964.8,4974.2
Exp/Cntr=0.3,0.1

Type RM Length L Ch R = 1,15543,451,451,451
BEGIN DESCRIPTION:
West Dry Branch 34.0
END DESCRIPTION:
XS GIS Cut Line= 3
      1868025.01     13976725.00      1867925.00     13976725.00
      1867299.05     13976872.45
#Sta/Elev= 30
  4900.1 2026.64  4902.6 2026.64  4930.1 2021.74  4950.1 2019.24  4970.1 2014.60
  4980.1 2008.44  4990.1 2004.96  4992.9 2001.94  4993.4 2001.44  5001.9 2001.44
  5002.4 2001.94  5018.7 2002.00  5041.2 2003.83  5066.2 2004.83  5072.0 2004.40
  5092.6 2005.25  5102.8 2006.53  5108.6 2006.29  5175.3 2009.15  5226.1 2011.15
  5330.6 2013.79  5367.8 2015.38  5390.5 2015.23  5410.2 2016.41  5431.6 2016.36
  5483.0 2018.07  5524.1 2020.63  5571.4 2022.28  5589.9 2022.78  5643.2 2025.67
#Mann=5,-1,0
  4900.1    0.07       0  4992.9    0.05       0  5002.4    0.07       0
  5175.3     0.1       0  5571.4    0.07       0
Bank Sta=4992.9,5002.4
Exp/Cntr=0.3,0.1

Type RM Length L Ch R = 1,15092,469,469,469
BEGIN DESCRIPTION:
West Dry Branch 33.0
END DESCRIPTION:
XS GIS Cut Line= 3
      1867875.02     13976274.99      1867775.00     13976325.00
      1867309.80     13976647.19
#Sta/Elev= 30
  4883.7 2021.50  4964.8 2010.96  4973.2 2008.53  4981.5 2000.98  4987.1 1996.55
  4987.9 1993.54  4988.4 1993.04  4997.0 1993.04  4997.5 1993.54  5009.0 1994.81
  5017.8 1997.32  5023.9 2000.09  5046.0 1999.84  5059.7 2001.04  5068.5 2000.71
  5089.4 2001.36  5146.2 2005.97  5190.2 2007.26  5203.0 2008.49  5214.3 2008.79
  5226.6 2010.32  5281.7 2011.27  5348.3 2014.16  5379.4 2016.23  5390.8 2016.39
  5404.4 2017.57  5498.2 2021.26  5527.9 2021.78  5544.4 2022.98  5561.4 2023.48
#Mann=9,-1,0
  4883.7     0.1       0  4987.9    0.05       0  4997.5     0.1       0
  5046.0    0.07       0  5214.3     0.1       0  5281.7   0.035       0
  5379.4     0.1       0  5404.4   0.035       0  5544.4    0.07       0
Bank Sta=4987.9,4997.5
Exp/Cntr=0.3,0.1

Type RM Length L Ch R = 1,14623,464,464,464
BEGIN DESCRIPTION:
West Dry Branch 32.0
END DESCRIPTION:
XS GIS Cut Line= 3
      1867525.03     13975974.99      1867425.00     13976025.00
      1867025.03     13976324.98
#Sta/Elev= 30
  4888.4 2012.80  4916.4 2010.88  4924.8 2009.56  4963.9 2001.85  4969.5 1998.28
  4991.8 1995.43  4992.6 1994.85  4993.1 1994.35  5001.7 1994.35  5002.2 1994.85
  5028.4 1995.21  5043.6 1996.35  5072.1 1995.70  5122.1 1999.15  5128.4 2000.41
  5136.7 2000.81  5142.9 2001.98  5166.1 2003.56  5207.5 2005.76  5213.8 2007.40
  5228.4 2008.83  5300.2 2012.61  5313.8 2014.18  5336.7 2015.30  5363.8 2018.81
  5392.9 2019.62  5436.7 2022.31  5450.2 2024.44  5468.0 2025.76  5500.2 2027.47
#Mann=6,-1,0
  4888.4    0.07       0  4992.6    0.05       0  5002.2    0.07       0
  5043.6     0.1       0  5166.1    0.07       0  5468.0   0.035       0
Bank Sta=4992.6,5002.2
Exp/Cntr=0.3,0.1

Type RM Length L Ch R = 1,14159,475,475,475
BEGIN DESCRIPTION:
West Dry Branch 31.0
END DESCRIPTION:
XS GIS Cut Line= 3
      1867325.01     13975725.00      1867025.00     13975825.00
      1866924.97     13975925.03
#Sta/Elev= 30
  4690.7 2010.77  4711.8 2010.71  4732.9 2010.00  4743.4 2008.95  4776.8 2006.82
  4785.6 2006.64  4796.1 2005.51  4827.7 2003.46  4838.3 2002.10  4848.8 2001.95
  4860.8 2001.29  4869.9 1999.79  4880.4 1999.45  4901.5 1996.90  4912.1 1996.12
  4933.1 1995.36  4943.7 1993.99  4975.3 1993.27  4985.9 1993.70  4999.5 1993.01
  5000.0 1992.51  5008.7 1992.51  5009.2 1993.01  5035.2 1993.53  5049.4 1994.96
  5063.5 2000.14  5077.6 2004.77  5105.9 2010.17  5134.2 2012.33  5148.4 2012.93
#Mann=5,-1,0
  4690.7     0.1       0  4776.8    0.07       0  4860.8     0.1       0
  4999.5    0.05       0  5009.2     0.1       0
Bank Sta=4999.5,5009.2
Exp/Cntr=0.3,0.1

Type RM Length L Ch R = 1,13684,456,456,456
BEGIN DESCRIPTION:
West Dry Branch 30.0
END DESCRIPTION:
XS GIS Cut Line= 3
      1867175.00     13975525.00      1866775.00     13975475.00
      1866675.01     13975475.00
#Sta/Elev= 30
  4596.8 2006.27  4606.9 2006.39  4639.6 2004.93  4657.3 2002.52  4667.3 2001.87
  4677.4 2002.16  4737.9 1998.61  4794.9 1996.79  4848.7 1995.17  4868.9 1993.84
  4876.5 1992.62  4881.5 1993.19  4893.8 1992.12  4949.5 1990.72  4962.1 1989.97
  4969.7 1988.38  4989.8 1987.73  4992.5 1986.96  4993.0 1986.46  5001.8 1986.46
  5002.3 1986.96  5019.9 1988.76  5029.9 1993.18  5039.9 2004.37  5049.9 2013.91
  5059.9 2017.36  5069.9 2019.45  5089.9 2021.98  5097.4 2024.47  5099.9 2024.47
#Mann=5,-1,0
  4596.8     0.1       0  4794.9    0.07       0  4893.8     0.1       0
  4992.5    0.05       0  5002.3     0.1       0
Bank Sta=4992.5,5002.3
Exp/Cntr=0.3,0.1

Type RM Length L Ch R = 1,13228,469,469,469
BEGIN DESCRIPTION:
West Dry Branch 29.0
END DESCRIPTION:
XS GIS Cut Line= 3
      1867225.00     13975275.00      1866925.00     13975075.00
      1866824.95     13975075.00
#Sta/Elev= 30
  4643.9 2006.94  4651.4 2006.24  4672.4 2005.54  4693.5 2004.11  4702.5 2002.93
  4708.5 2002.70  4729.5 2000.67  4752.1 1997.57  4759.6 1996.15  4837.7 1990.32
  4867.7 1988.82  4882.8 1988.77  4909.8 1987.10  4932.3 1987.35  4945.9 1986.13
  4960.9 1985.60  4968.4 1983.60  4975.9 1983.32  4981.9 1981.98  4990.9 1980.99
  4996.5 1979.62  4997.0 1979.12  5005.9 1979.12  5006.4 1979.62  5014.5 1980.96
  5038.0 1997.62  5044.5 2002.29  5054.5 2006.96  5064.5 2010.89  5104.5 2013.28
#Mann=4,-1,0
  4643.9     0.1       0  4996.5    0.05       0  5006.4     0.1       0
  5038.0    0.07       0
Bank Sta=4996.5,5006.4
Exp/Cntr=0.3,0.1

Type RM Length L Ch R = 1,12759,459,459,459
BEGIN DESCRIPTION:
West Dry Branch 28.0
END DESCRIPTION:
XS GIS Cut Line= 3
      1867475.01     13974925.01      1867275.00     13974775.00
      1867124.99     13974674.99
#Sta/Elev= 30
  4750.0 2007.03  4786.5 2006.35  4807.3 2004.34  4842.7 1997.10  4863.6 1994.99
  4878.1 1992.73  4892.7 1988.75  4900.0 1985.85  4913.6 1981.94  4936.5 1981.95
  4942.7 1981.36  4963.6 1981.66  4986.5 1979.38  4991.9 1978.37  4992.4 1977.87
  5001.4 1977.87  5001.9 1978.37  5013.5 1980.60  5022.5 1981.23  5028.6 1983.19
  5036.1 1982.93  5049.6 1986.45  5058.6 1988.13  5064.6 1990.34  5100.7 1998.27
  5115.7 2002.30  5151.7 2009.30  5157.8 2009.58  5166.8 2011.07  5180.3 2011.32
#Mann=3,-1,0
  4750.0     0.1       0  4991.9    0.05       0  5001.9     0.1       0
Bank Sta=4991.9,5001.9
Exp/Cntr=0.3,0.1

Type RM Length L Ch R = 1,12300,445,445,445
BEGIN DESCRIPTION:
West Dry Branch 27.0
END DESCRIPTION:
XS GIS Cut Line= 3
      1867724.96     13974525.00      1867625.00     13974525.00
      1867275.04     13974375.02
#Sta/Elev= 30
  4891.2 2006.84  4893.7 2006.84  4921.2 2002.29  4931.2 1999.72  4961.2 1994.26
  4971.2 1991.41  4981.2 1985.70  4988.7 1978.43  4993.9 1978.43  5000.2 1974.83
  5007.9 1973.81  5008.4 1973.31  5017.5 1973.31  5018.0 1973.81  5023.8 1974.03
  5034.7 1976.42  5076.4 1980.86  5081.8 1980.29  5089.1 1981.19  5100.0 1981.39
  5134.4 1980.31  5152.5 1980.63  5165.2 1982.26  5187.0 1986.76  5219.6 1990.50
  5241.4 1994.14  5274.0 1996.92  5317.6 2003.17  5354.4 2005.53  5371.9 2005.99
#Mann=4,-1,0
  4891.2     0.1       0  5007.9    0.05       0  5018.0     0.1       0
  5354.4    0.07       0
Bank Sta=5007.9,5018
Exp/Cntr=0.3,0.1

Type RM Length L Ch R = 1,11855,450,450,450
BEGIN DESCRIPTION:
West Dry Branch 26.0
END DESCRIPTION:
XS GIS Cut Line= 3
      1867875.05     13974125.00      1867775.00     13974125.00
      1867474.98     13974175.00
#Sta/Elev= 30
  4894.9 2009.62  4897.4 2009.62  4904.9 2008.49  4914.9 2006.51  4954.9 1991.85
  4964.9 1987.76  4974.9 1982.51  4984.9 1978.85  4992.4 1969.49  4997.5 1969.49
  5000.0 1967.51  5000.5 1967.01  5009.6 1967.01  5010.1 1967.51  5035.5 1967.97
  5045.6 1971.52  5055.8 1974.01  5076.0 1975.86  5106.5 1977.41  5167.3 1978.76
  5177.4 1979.27  5197.7 1981.38  5205.3 1982.64  5210.4 1982.58  5228.1 1985.91
  5238.3 1987.19  5266.1 1989.59  5271.2 1989.46  5296.5 1991.95  5299.1 1991.95
#Mann=3,-1,0
  4894.9    0.07       0  5000.0    0.05       0  5010.1    0.07       0
Bank Sta=5000,5010.1
Exp/Cntr=0.3,0.1

Type RM Length L Ch R = 1,11405,467,467,467
BEGIN DESCRIPTION:
West Dry Branch 25.0
END DESCRIPTION:
XS GIS Cut Line= 3
      1867875.00     13973675.00      1867775.00     13973675.00
      1867375.01     13973875.00
#Sta/Elev= 30
  4896.3 2003.03  4898.8 2003.03  4906.3 1999.73  4926.3 1994.05  4946.3 1984.30
  4966.3 1976.31  4976.3 1971.06  4986.3 1969.09  4993.8 1969.84  5004.7 1969.79
  5018.7 1968.77  5041.0 1969.85  5066.5 1968.60  5067.0 1968.10  5076.5 1968.10
  5077.0 1968.60  5099.7 1969.74  5116.5 1973.22  5130.5 1974.67  5175.2 1977.00
  5211.5 1977.59  5219.9 1978.20  5233.9 1977.99  5303.8 1982.77  5340.1 1984.18
  5345.7 1985.00  5354.1 1985.34  5390.4 1988.79  5435.1 1991.55  5443.5 1992.46
#Mann=3,-1,0
  4896.3    0.07       0  5066.5    0.05       0  5077.0    0.07       0
Bank Sta=5066.5,5077
Exp/Cntr=0.3,0.1

Type RM Length L Ch R = 1,10938,465,465,465
BEGIN DESCRIPTION:
West Dry Branch 24.0
END DESCRIPTION:
XS GIS Cut Line= 3
      1867624.97     13973275.02      1867525.00     13973325.00
      1867124.98     13973375.00
#Sta/Elev= 30
  4892.8 1991.85  4906.7 1990.24  4915.1 1988.60  4929.1 1985.61  4959.8 1977.79
  4968.5 1961.62  4969.0 1961.12  4978.6 1961.12  4979.1 1961.62  4996.2 1962.30
  5007.1 1961.77  5034.8 1962.84  5047.4 1964.72  5115.4 1968.23  5128.0 1969.86
  5186.0 1971.21  5203.6 1972.75  5246.4 1979.74  5276.7 1985.58  5284.2 1988.33
  5306.9 1993.28  5327.1 1997.06  5337.1 2000.25  5357.3 2005.34  5364.9 2008.45
  5369.9 2008.73  5377.4 2011.51  5387.5 2013.78  5397.6 2015.20  5407.7 2015.27
#Mann=3,-1,0
  4892.8    0.07       0  4968.5    0.05       0  4979.1    0.07       0
Bank Sta=4968.5,4979.1
Exp/Cntr=0.3,0.1

Type RM Length L Ch R = 1,10473,477,477,477
BEGIN DESCRIPTION:
West Dry Branch 23.0
END DESCRIPTION:
XS GIS Cut Line= 3
      1867575.00     13973125.00      1867225.00     13972975.00
      1867124.99     13972975.00
#Sta/Elev= 30
  4625.0 1980.26  4646.8 1979.05  4679.4 1978.43  4733.8 1972.87  4768.3 1970.53
  4782.4 1970.22  4844.4 1969.10  4862.5 1966.69  4868.0 1967.30  4897.0 1963.13
  4915.1 1958.98  4920.6 1960.22  4929.6 1957.69  4944.1 1957.83  4973.2 1956.19
  4996.7 1956.58  4997.8 1956.05  4998.3 1955.55  5007.9 1955.55  5008.4 1956.05
  5015.8 1957.06  5025.8 1960.96  5032.6 1964.29  5045.8 1972.08  5055.8 1978.93
  5065.8 1984.36  5075.8 1991.70  5095.8 2001.81  5103.3 2007.45  5105.8 2007.45
#Mann=5,-1,0
  4625.0    0.07       0  4782.4   0.035       0  4997.8   0.035       0
  5008.4   0.035       0  5032.6    0.07       0
Bank Sta=4997.8,5008.4
Exp/Cntr=0.3,0.1

Type RM Length L Ch R = 1,9996,467,467,467
BEGIN DESCRIPTION:
West Dry Branch 22.0
END DESCRIPTION:
XS GIS Cut Line= 3
      1867824.97     13972974.97      1867525.00     13972675.00
      1867425.03     13972575.03
#Sta/Elev= 30
  4575.8 1994.26  4589.9 1993.86  4604.0 1992.71  4618.2 1992.17  4632.3 1990.47
  4646.5 1987.27  4660.6 1985.09  4703.0 1979.91  4717.2 1978.58  4745.5 1973.07
  4759.6 1971.11  4773.7 1968.39  4787.9 1966.85  4858.6 1959.83  4957.6 1956.19
  4971.7 1954.43  4985.9 1949.88  4996.5 1948.40  5003.6 1948.40  5008.8 1947.37
  5009.3 1946.87  5019.0 1946.87  5019.5 1947.37  5035.4 1951.71  5042.4 1962.06
  5070.7 1980.92  5084.9 1986.34  5099.0 1992.92  5127.3 1998.57  5141.4 1998.98
#Mann=3,-1,0
  4575.8    0.07       0  5008.8    0.05       0  5019.5    0.07       0
Bank Sta=5008.8,5019.5
Exp/Cntr=0.3,0.1

Type RM Length L Ch R = 1,9529,465,465,465
BEGIN DESCRIPTION:
West Dry Branch 21.0
END DESCRIPTION:
XS GIS Cut Line= 3
      1868074.98     13972574.99      1867925.00     13972475.00
      1867524.96     13972374.99
#Sta/Elev= 30
  4818.4 1999.97  4831.9 1998.09  4854.4 1991.39  4861.9 1986.54  4877.0 1980.56
  4898.0 1965.81  4904.0 1959.48  4913.0 1954.87  4919.0 1947.95  4926.5 1946.03
  4934.1 1945.30  4934.7 1941.94  4935.2 1941.44  4945.5 1941.94  4976.1 1945.88
  4985.1 1946.10  4995.6 1948.10  5063.1 1948.57  5091.4 1952.12  5112.0 1955.92
  5153.3 1960.24  5186.8 1962.71  5228.0 1967.70  5246.0 1970.15  5264.1 1975.42
  5269.2 1975.56  5277.0 1977.65  5310.5 1980.44  5380.0 1991.49  5411.0 1992.55
#Mann=3,-1,0
  4818.4    0.07       0  4934.7    0.05       0  4945.5    0.07       0
Bank Sta=4934.7,4945.5
Exp/Cntr=0.3,0.1
