--- North Creek.prj (project) ---

Proj Title=North Creek Base Level Engineering
Current Plan=p01
Default Exp/Contr=0.3,0.1
English Units
Geom File=g01
Flow File=f01
Plan File=p01
Y Axis Title=Elevation
X Axis Title(PF)=Main Channel Distance
X Axis Title(XS)=Station
BEGIN DESCRIPTION:
North Creek
END DESCRIPTION:
DSS Export Rating Curves= 0
DSS Export Rating Curve Sorted= 0
DSS Export Volume Flow Curves= 0
DXF OffsetX= 0
DXF OffsetY= 0
DXF ScaleX= 1
DXF ScaleY= 10

--- North Creek.p01 (plan) ---

Plan Title=Multiple Run
Short Identifier=Multiple
Geom File=g01
Flow File=f01
Subcritical Flow
K Sum by GR= 0
Std Step Tol= 0.01
Critical Tol= 0.01
Num of Std Step Trials= 20
Max Error Tol= 0.3
Flow Tol Ratio= 0.001
Split Flow NTrial= 30
Split Flow Tol= 0.02
Split Flow Ratio= 0.02
Log Output Level= 0
Friction Slope Method= 1
Unsteady Friction Slope Method= 2
Unsteady Bridges Friction Slope Method= 1
Parabolic Critical Depth
Global Vel Dist=  1 , 1 , 1
Global Log Level= 0
CheckData=True
Encroach Param= -1, 0, 0, 0
BEGIN DESCRIPTION:
Multiple Run
END DESCRIPTION:

--- North Creek.f01 (steady flow) ---

Flow Title=Multiple
Program Version=4.10
Number of Profiles= 7
Profile Names=10-year,25-year,50-year,1pct_min,100-year,1pct_plu,500-year
River Rch & RM=North Creek,Reach-1         ,51283
     612    1024    1411     947    1889    3768    3349
River Rch & RM=North Creek,Reach-1         ,46231
     994    1707    2393    1629    3251    6487    5949
River Rch & RM=North Creek,Reach-1         ,41178
    1515    2657    3778    2603    5195   10364    9746
River Rch & RM=North Creek,Reach-1         ,36450
    2327    4159    5991    4175    8329   16619   15989
River Rch & RM=North Creek,Reach-1         ,31534
    3154    5712    8300    5828   11629   23202   22675
River Rch & RM=North Creek,Reach-1         ,28225
    3842    7015   10249    7232   14429   28790   28408
River Rch & RM=North Creek,Reach-1         ,25936
    3921    7157   10455    7374   14714   29358   28951
River Rch & RM=North Creek,Reach-1         ,24153
    4354    7973   11670    8246   16452   32826   32481
River Rch & RM=North Creek,Reach-1         ,21242
    4672    8541   12490    8816   17591   35098   34644
River Rch & RM=North Creek,Reach-1         ,19328
    4846    8854   12944    9130   18218   36349   35832
River Rch & RM=North Creek,Reach-1         ,14352
    4980    9104   13313    9393   18742   37396   36880
River Rch & RM=North Creek,Reach-1         ,13113
    5463    9985   14599   10294   20539   40981   40365
River Rch & RM=North Creek,Reach-1         ,2459
    6743   12397   18192   12853   25645   51169   50514
Boundary for River Rch & Prof#=North Creek,Reach-1         , 1
Up Type= 0
Dn Type= 3
Dn Slope=0.006
Boundary for River Rch & Prof#=North Creek,Reach-1         , 2
Up Type= 0
Dn Type= 3
Dn Slope=0.006
Boundary for River Rch & Prof#=North Creek,Reach-1         , 3
Up Type= 0
Dn Type= 3
Dn Slope=0.006
Boundary for River Rch & Prof#=North Creek,Reach-1         , 4
Up Type= 0
Dn Type= 3
Dn Slope=0.006
Boundary for River Rch & Prof#=North Creek,Reach-1         , 5
Up Type= 0
Dn Type= 3
Dn Slope=0.006
Boundary for River Rch & Prof#=North Creek,Reach-1         , 6
Up Type= 0
Dn Type= 3
Dn Slope=0.006
Boundary for River Rch & Prof#=North Creek,Reach-1         , 7
Up Type= 0
Dn Type= 3
Dn Slope=0.006
DSS Import GetInterval= 0
DSS Import GetPeak= 0
DSS Import FillOption= 0

--- North Creek.g01 (geometry) ---

Geom Title=Existing Conditions
Program Version=4.10

River Reach=North Creek     ,Reach-1
Reach XY= 30
        1991875.       13944975.      1991661.53     13944211.43
      1990627.07     13943419.14      1990577.06     13942580.85
      1990975.24     13942050.08      1990725.24     13941240.22
      1991771.96     13939223.58      1991730.08     13938272.69
      1992264.53     13938084.83      1992234.13     13937618.22
      1992664.37       13937535.      1993422.75     13936119.07
      1993375.07     13932240.39      1993935.65       13931065.
      1994423.95     13930864.58      1994377.26     13927280.94
      1995819.17      13925777.3      1996104.58     13924344.77
      1997915.87     13923731.72      1997277.17     13922480.97
      1998128.83     13919426.58      1999425.55     13917464.81
      1997783.16     13915381.05      1997319.48     13914022.57
      1995530.84     13911377.29      1995319.46     13909922.58
      1994030.48     13908677.44      1993967.19     13907568.81
      1992197.88     13906698.52        1991525.       13905075.

Type RM Length L Ch R = 1 ,51283   ,448,448,448
BEGIN DESCRIPTION:
North Creek 105.0
END DESCRIPTION:
XS GIS Cut Line= 3
        1991975.       13944625.        1991825.       13944675.
      1991725.01     13944724.99
#Sta/Elev= 30
  4846.2 2073.11  4850.4 2072.79  4856.7 2071.09  4869.3 2068.53  4872.5 2067.38
  4876.9 2066.58  4880.5 2065.42    4901 2059.21  4907.3 2056.78  4913.6 2055.26
  4916.8 2054.05  4938.9 2047.64  4957.9 2040.25  4971.8  2035.3    4980 2031.86
  4984.3 2030.84  4984.6 2030.34  4988.1 2030.34  4988.3 2030.84  4990.7 2031.78
    4999 2033.93    5016 2041.12  5028.9 2045.82  5069.1 2059.43  5072.5 2059.97
  5085.9 2064.07  5092.6 2065.65  5095.9 2065.97  5112.7 2069.44  5116.1 2069.56
#Mann= 4 ,-1 , 0
  4846.2    .035       0  4880.5     .07       0  4984.3     .05       0
  4988.3     .07       0
Bank Sta=4984.3,4988.3
XS Rating Curve= 0 ,0
Exp/Cntr=0.3,0.1

Type RM Length L Ch R = 1 ,50835   ,217,217,217
BEGIN DESCRIPTION:
North Creek 104.0
END DESCRIPTION:
XS GIS Cut Line= 3
      1991774.99     13944225.01        1991675.       13944275.
        1991625.       13944325.
#Sta/Elev= 30
  4892.8 2037.24  4903.3 2034.81  4911.2 2033.85  4915.6 2032.45  4921.8 2031.66
  4925.2 2030.72  4935.2 2028.97  4936.9 2028.44  4944.7 2025.38    4947 2024.98
  4948.6 2024.39  4962.1 2017.88  4968.8 2014.92  4978.8  2009.9  4986.9 2006.82
  4987.1 2006.32  4990.6 2006.32  4990.9 2006.82    4999 2009.67  5010.2 2015.91
  5016.9 2018.43  5021.2 2020.43  5029.6  2023.8  5030.5 2024.39  5035.6 2026.19
  5039.9 2027.46  5044.1 2028.15  5050.8 2029.92  5061.1 2032.04  5075.3 2034.49
#Mann= 3 ,-1 , 0
  4892.8     .07       0  4986.9     .05       0  4990.9     .07       0
Bank Sta=4986.9,4990.9
XS Rating Curve= 0 ,0
Exp/Cntr=0.3,0.1

Type RM Length L Ch R = 1 ,50618   ,203,203,203
BEGIN DESCRIPTION:
Mapping XS f594865e
END DESCRIPTION:
XS GIS Cut Line= 2
      1991585.59     13944059.43      1991417.86     13944322.27
#Sta/Elev= 30
  4907.7 2032.44    4930 2027.69    4944 2022.98  4953.3 2019.18  4971.9 2011.89
  4985.1 2007.26  4988.8 2005.39  4997.4 2003.21  4999.8 2002.22  5011.5 1999.63
  5014.8 1998.94  5015.2 1998.45  5015.4 1997.95  5018.9 1997.95  5019.2 1998.45
  5022.1 1999.24  5027.8    2002  5040.8  2006.9  5044.4 2008.67  5049.2 2010.01
  5052.8 2011.75  5061.2 2013.94  5067.7 2016.25  5072.3 2018.15  5091.9 2023.32
  5116.9 2028.96  5161.5 2033.91    5182 2037.59    5195 2038.85  5219.5 2043.45
#Mann= 6 ,-1 , 0
  4907.7      .1       0  4953.3     .07       0  5011.5    .035       0
  5015.2     .05       0  5019.2    .035       0  5067.7     .07       0
Bank Sta=5015.2,5019.2
XS Rating Curve= 0 ,0
Exp/Cntr=0.3,0.1

Type RM Length L Ch R = 1 ,50415   ,473,473,473
BEGIN DESCRIPTION:
North Creek 103.0
END DESCRIPTION:
XS GIS Cut Line= 3
      1991524.98     13943975.01        1991375.       13944025.
        1991325.       13944125.
#Sta/Elev= 30
  4841.9 2033.59  4871.4 2028.18    4878 2026.14    4897 2021.72  4909.5 2017.38
  4918.8 2014.09  4936.1  2009.6  4953.6 2005.32  4973.8 1999.43  4985.2 1993.69
  4992.7 1991.83  4992.9 1991.33  4996.4 1991.33  4996.7 1991.83  5004.1 1994.43
  5014.2 1996.57  5020.9 1998.82  5034.3 2004.89  5037.7 2005.95  5044.4 2009.94
  5057.8  2014.7  5062.5 2017.54  5067.9 2019.18  5071.2 2020.91  5081.3  2024.7
  5084.6 2025.43  5092.1 2029.29  5101.4 2031.09  5108.1 2032.93  5111.8  2033.4
#Mann= 6 ,-1 , 0
  4841.9      .1       0  4909.5    .035       0  4936.1     .07       0
  4992.7     .05       0  4996.7     .07       0  5092.1    .035       0
Bank Sta=4992.7,4996.7
XS Rating Curve= 0 ,0
Exp/Cntr=0.3,0.1

Type RM Length L Ch R = 1 ,49942   ,418,418,418
BEGIN DESCRIPTION:
North Creek 102.0
END DESCRIPTION:
XS GIS Cut Line= 3
      1991074.99     13943675.02        1990975.       13943825.
        1990975.     13944025.04
#Sta/Elev= 30
  4819.7 2025.54  4832.2 2022.57  4863.9 2013.21  4880.9  2009.1  4897.1 2003.99
  4905.9 2002.47  4916.7 1999.35  4956.5 1986.08  4970.8  1979.5  4984.6 1975.13
  4988.8 1973.05  4999.6 1970.86  5012.7 1970.34  5012.9 1969.84  5016.7 1970.34
  5022.3  1972.5  5035.7  1976.4  5041.6 1979.84  5044.7 1980.47  5053.6 1984.11
  5056.7 1986.52  5059.7 1987.57  5065.7 1991.31  5077.7  1995.6  5083.7 1998.67
  5092.7 2000.98  5122.6 2011.25  5156.1  2024.2  5164.7 2027.17    5200 2033.75
#Mann= 6 ,-1 , 0
  4819.7      .1       0  4863.9     .07       0  5012.7     .05       0
  5016.7     .07       0  5022.3    .035       0  5156.1     .07       0
Bank Sta=5012.7,5016.7
XS Rating Curve= 0 ,0
Exp/Cntr=0.3,0.1

Type RM Length L Ch R = 1 ,49524   ,225,225,225
BEGIN DESCRIPTION:
North Creek 101.0
END DESCRIPTION:
XS GIS Cut Line= 3
      1990775.01       13943525.        1990725.       13943525.
      1990625.03     13943624.97
#Sta/Elev= 30
  4945.2 1978.17  4967.2 1971.56  4975.5 1970.01  4979.2 1969.61  4982.2 1968.56
  4985.2 1965.68  4988.2 1961.87  4991.2 1960.26    4998 1957.52  5002.2 1954.87
  5006.5 1953.25  5013.5 1951.48  5013.7 1950.98  5017.2 1950.98  5017.5 1951.48
  5027.7 1954.35  5031.9 1956.59  5037.2 1958.74  5040.9 1962.66  5044.7 1967.97
  5045.7 1968.55  5054.2 1969.96  5075.4  1976.1  5079.7 1976.94  5088.1 1980.01
  5092.4 1981.06  5096.6 1981.62  5108.3 1984.71    5121 1986.75  5136.6 1988.72
#Mann= 4 ,-1 , 0
  4945.2      .1       0  4975.5     .07       0  5013.5     .05       0
  5017.5     .07       0
Bank Sta=5013.5,5017.5
XS Rating Curve= 0 ,0
Exp/Cntr=0.3,0.1

Type RM Length L Ch R = 1 ,49299   ,230,230,230
BEGIN DESCRIPTION:
Mapping XS 0f06c7dc
END DESCRIPTION:
XS GIS Cut Line= 2
      1990847.12     13943268.77      1990406.04     13943408.89
#Sta/Elev= 30
  4766.8 2013.94  4862.4 1990.16  4890.2 1982.24  4900.1 1978.31  4903.3 1977.83
    4910 1975.37  4923.7 1971.56  4929.2 1970.92  4931.6 1970.69  4934.8 1969.19
  4937.9 1965.52  4941.1 1959.52  4961.9 1949.76  4975.7 1944.73  4991.1 1940.85
  4991.3 1940.35  4994.8 1940.35  4995.1 1940.85    5004 1943.41  5019.8 1952.88
  5032.3 1962.07  5041.8 1966.61  5044.9 1970.08  5057.7  1972.9  5076.4 1979.18
  5101.6 1985.28  5156.3 1995.87  5186.6 1999.28  5202.3  2002.1  5229.6 2005.62
#Mann= 4 ,-1 , 0
  4766.8      .1       0  4929.2     .07       0  4991.1     .05       0
  4995.1     .07       0
Bank Sta=4991.1,4995.1
XS Rating Curve= 0 ,0
Exp/Cntr=0.3,0.1

Type RM Length L Ch R = 1 ,49069   ,260,260,260
BEGIN DESCRIPTION:
North Creek 100.0
END DESCRIPTION:
XS GIS Cut Line= 3
      1990725.01       13943125.        1990575.       13943125.
      1990474.99     13943275.01
#Sta/Elev= 30
  4849.3 1977.94  4857.3 1975.76  4890.3 1971.46  4896.3 1968.31  4898.6 1960.57
  4899.3 1959.26  4901.6 1958.99  4902.3 1958.25  4908.3 1956.42  4926.3 1947.84
  4930.7 1946.56  4949.6 1940.34  4953.3 1938.48  4964.6 1935.77  4971.3 1934.92
  4978.3 1932.91  4978.5 1932.41    4982 1932.41  4982.3 1932.91  5007.7 1933.06
  5009.9 1933.58  5021.8 1939.85  5029.9 1942.75  5054.2 1948.96  5062.3  1950.4
  5100.2 1962.48  5115.5 1965.88  5127.2  1972.5  5148.9 1974.33  5179.6 1979.92
#Mann= 4 ,-1 , 0
  4849.3      .1       0  4930.7     .07       0  4978.3     .05       0
  4982.3     .07       0
Bank Sta=4978.3,4982.3
XS Rating Curve= 0 ,0
Exp/Cntr=0.3,0.1

Type RM Length L Ch R = 1 ,48809   ,240,240,240
BEGIN DESCRIPTION:
Mapping XS 0f425970
END DESCRIPTION:
XS GIS Cut Line= 2
      1990800.49     13942866.27      1990328.79     13942864.06
#Sta/Elev= 30
  4774.5 2002.59  4821.9 1992.36  4827.9 1991.72  4842.9 1986.18  4854.9 1982.92
  4869.9 1976.68  4881.9 1973.17  4884.9 1969.93  4890.9 1968.44  4899.9 1963.19
  4923.9 1953.14  4950.9 1940.55  4962.9 1933.94  4974.9 1928.57  4980.9 1926.69
    4993 1924.75  4999.5 1921.58    5000 1920.56  5000.2 1920.06    5004 1920.56
    5020  1926.1    5047 1942.24    5056 1945.41  5080.1 1957.72    5092 1962.57
    5101 1973.56  5109.9 1975.21  5130.8 1982.19    5146 1986.09  5246.2  2004.7
#Mann= 4 ,-1 , 0
  4774.5      .1       0  4950.9     .07       0    5000     .05       0
    5004     .07       0
Bank Sta=5000,5004
XS Rating Curve= 0 ,0
Exp/Cntr=0.3,0.1

Type RM Length L Ch R = 1 ,48569   ,447,447,447
BEGIN DESCRIPTION:
North Creek 99.0
END DESCRIPTION:
XS GIS Cut Line= 3
      1990774.95     13942674.99        1990575.       13942625.
      1990375.01     13942724.99
#Sta/Elev= 30
  4793.4 1987.67  4834.5 1976.99  4846.9 1974.71  4850.5 1971.74  4852.9 1966.89
  4857.9 1963.41  4870.2 1957.61  4877.7 1955.56  4880.9 1953.55  4904.9 1944.22
  4913.4 1941.86    4937 1932.22  4951.2 1924.67  4984.1 1913.08  4984.3 1912.58
  4988.1 1913.08  4995.3 1918.07  5011.8 1920.52  5062.1  1937.7  5088.9 1944.44
  5115.7 1953.13  5139.7  1963.1  5145.9 1966.79  5149.3 1971.56  5152.6 1973.25
  5159.3 1973.29  5166.1 1974.56  5192.9  1981.6  5202.9    1986  5223.1 1989.13
#Mann= 4 ,-1 , 0
  4793.4      .1       0  4913.4     .07       0  4984.1     .05       0
  4988.1     .07       0
Bank Sta=4984.1,4988.1
XS Rating Curve= 0 ,0
Exp/Cntr=0.3,0.1

Type RM Length L Ch R = 1 ,48122   ,471,471,471
BEGIN DESCRIPTION:
North Creek 98.0
END DESCRIPTION:
XS GIS Cut Line= 3
      1990974.99     13942424.99        1990825.       13942275.
      1990775.02     13942225.02
#Sta/Elev= 30
  4792.7 1995.88  4806.3 1992.23  4848.7 1978.01  4850.9 1975.09    4853  1970.1
  4858.2 1966.14  4876.3 1957.59    4886 1952.14  4900.6 1945.77  4907.2  1941.5
  4934.5 1929.38  4952.7 1920.11  4965.4 1912.55  4970.8 1910.61    4976 1907.21
  4981.2 1905.23  4988.7 1898.92  4996.2 1894.09  4996.4 1893.59  5000.2 1894.09
  5003.6 1894.53  5006.6 1895.84  5012.1 1900.33  5023.6 1906.86  5030.2 1909.84
  5035.4 1914.01  5041.8 1917.59  5050.3 1923.48    5063 1927.15  5075.5 1933.11
#Mann= 3 ,-1 , 0
  4792.7     .07       0  4996.2     .05       0  5000.2     .07       0
Bank Sta=4996.2,5000.2
XS Rating Curve= 0 ,0
Exp/Cntr=0.3,0.1

Type RM Length L Ch R = 1 ,47651   ,481,481,481
BEGIN DESCRIPTION:
North Creek 97.0
END DESCRIPTION:
XS GIS Cut Line= 3
      1991074.98       13941875.        1990925.       13941875.
      1990825.08       13941875.
#Sta/Elev= 30
  4854.6  1924.7  4858.8 1923.93  4861.8 1922.79  4882.5 1918.58  4885.5 1917.08
  4912.8 1909.51  4926.9 1904.44  4942.5 1898.64  4957.5 1891.95  4963.8 1889.72
  4975.5 1886.83  5002.5 1881.09  5005.8 1879.17  5006.8  1876.5  5007.1    1876
  5010.6    1876  5010.8  1876.5  5020.5  1877.6  5029.5 1886.72  5032.5 1889.12
  5047.5 1895.45  5053.8 1898.72  5062.5 1904.04  5071.8  1908.9  5080.8 1914.52
  5086.5 1918.79  5092.5 1922.07  5095.5 1923.43  5101.5 1924.24  5104.5 1925.33
#Mann= 4 ,-1 , 0
  4854.6      .1       0  4926.9     .07       0  5006.8     .05       0
  5010.8     .07       0
Bank Sta=5006.8,5010.8
XS Rating Curve= 0 ,0
Exp/Cntr=0.3,0.1

Type RM Length L Ch R = 1 ,47170   ,476,476,476
BEGIN DESCRIPTION:
North Creek 96.0
END DESCRIPTION:
XS GIS Cut Line= 3
      1991074.96     13941375.01        1990825.       13941425.
      1990574.97     13941525.01
#Sta/Elev= 30
  4740.8 1978.01  4772.3 1974.41  4790.7 1961.47  4812.1 1950.58  4836.6 1941.74
  4851.9  1934.1    4866 1929.16  4904.3 1912.13  4928.4 1898.08    4937 1894.26
  4949.8  1888.1  4965.1 1878.51  5000.1 1863.66  5000.4 1863.16  5004.1 1863.66
  5011.8 1869.15  5021.5 1871.12    5070 1869.82  5086.1 1870.46  5101.3 1873.15
  5115.2 1877.74  5132.3 1886.76    5154 1900.92  5163.9 1909.92  5170.2 1913.33
  5179.8 1922.74  5199.2  1935.7  5208.9 1940.08    5238 1951.73    5265 1959.92
#Mann= 6 ,-1 , 0
  4740.8      .1       0    4937     .07       0  5000.1     .05       0
  5004.1     .07       0  5101.3    .035       0  5208.9     .07       0
Bank Sta=5000.1,5004.1
XS Rating Curve= 0 ,0
Exp/Cntr=0.3,0.1

Type RM Length L Ch R = 1 ,46694   ,463,463,463
BEGIN DESCRIPTION:
North Creek 95.0
END DESCRIPTION:
XS GIS Cut Line= 3
        1991025.       13941125.        1990825.       13941025.
      1990574.97     13940824.98
#Sta/Elev= 30
  4776.5 1941.39    4805 1932.04  4818.9 1925.39    4852 1913.04  4930.2 1878.73
  4949.7 1869.51  4983.9 1858.91  4990.6  1855.4  4997.3 1850.58    5004  1847.7
  5004.2  1847.2    5008  1847.7  5013.4 1851.85  5019.3 1854.68  5025.2 1855.38
  5041.3 1854.76  5063.6 1854.73  5066.2 1853.95  5072.1 1849.95  5076.4 1848.39
  5084.9 1851.58  5105.3 1862.79  5119.2  1867.9  5153.7 1883.93  5168.2 1889.05
  5176.7 1892.91  5262.1 1922.22  5289.8 1930.26  5300.5 1932.47  5320.3 1936.77
#Mann= 6 ,-1 , 0
  4776.5      .1       0    5004     .05       0    5008      .1       0
  5041.3     .07       0  5105.3      .1       0  5300.5     .07       0
Bank Sta=5004,5008
XS Rating Curve= 0 ,0
Exp/Cntr=0.3,0.1

Type RM Length L Ch R = 1 ,46231   ,450,450,450
BEGIN DESCRIPTION:
North Creek 94.0
END DESCRIPTION:
XS GIS Cut Line= 3
      1991175.02     13940775.01        1990875.       13940575.
        1990775.       13940475.
#Sta/Elev= 30
  4644.1 1943.36  4689.7 1930.47  4709.2 1922.67  4722.2 1919.39  4736.6 1913.96
  4740.2 1911.88  4767.6 1902.79  4805.1 1885.39  4830.3 1876.33    4865  1862.3
  4882.3 1857.48  4916.9 1850.88  4934.9  1844.5  4970.9 1844.33  4979.6 1842.48
  4992.6  1841.5  4999.3  1838.1  4999.5  1837.6  5003.3  1838.1  5007.5 1839.82
  5011.9 1845.88  5020.6  1848.5  5037.4 1856.09  5058.8 1867.17  5066.8 1872.63
  5071.3 1874.04  5092.5 1884.54  5113.5 1890.99    5122 1892.54  5146.1 1900.42
#Mann= 3 ,-1 , 0
  4644.1     .07       0  4999.3     .05       0  5003.3     .07       0
Bank Sta=4999.3,5003.3
XS Rating Curve= 0 ,0
Exp/Cntr=0.3,0.1

Type RM Length L Ch R = 1 ,45781   ,446,446,446
BEGIN DESCRIPTION:
North Creek 93.0
END DESCRIPTION:
XS GIS Cut Line= 3
      1991429.69     13940475.45        1991125.       13940225.
      1990975.07     13940025.09
#Sta/Elev= 30
  4610.2 1943.28  4682.2 1924.06  4693.9 1922.67  4746.9 1908.54  4763.8 1905.69
  4795.9 1895.14  4811.4 1887.57  4814.3 1885.57    4822 1875.68    4857 1853.39
    4879 1840.25  4894.4 1836.06  4913.1 1835.16  4949.4 1836.44  4967.3  1832.2
  4979.3 1831.57  4979.5 1831.07  4983.3 1831.57  4987.7 1834.86  4990.9 1841.75
    4992 1842.52  5008.7 1843.28  5016.2 1840.26  5023.7 1843.26    5035 1845.13
  5049.8 1845.15    5065 1847.57  5143.7 1871.46    5230  1901.8  5254.5  1908.1
#Mann= 4 ,-1 , 0
  4610.2      .1       0  4894.4     .07       0  4979.3     .05       0
  4983.3     .07       0
Bank Sta=4979.3,4983.3
XS Rating Curve= 0 ,0
Exp/Cntr=0.3,0.1

Type RM Length L Ch R = 1 ,45335   ,450,450,450
BEGIN DESCRIPTION:
North Creek 92.0
END DESCRIPTION:
XS GIS Cut Line= 3
      1991612.23     13939997.73        1991275.       13939925.
      1991025.04     13939825.02
#Sta/Elev= 30
  4654.5 1917.32  4680.3 1915.52  4711.9 1908.03  4769.3 1887.53  4796.9  1878.4
  4839.9 1861.77  4848.2  1859.6  4855.8 1856.39  4873.8 1850.77  4916.6 1842.69
  4936.6 1838.22  4944.2 1836.22  4962.6 1829.46  4979.5 1826.34    4982 1826.71
  4990.2 1825.19  4997.7 1824.84  4997.9 1824.34  5001.7 1824.84  5025.3 1826.74
  5073.8 1837.76  5093.1 1845.24  5117.4 1857.32  5135.8 1865.35  5154.5 1872.42
  5177.2 1882.35  5199.8  1893.8  5222.4 1903.85  5261.2 1916.19  5268.7 1917.59
#Mann= 3 ,-1 , 0
  4654.5     .07       0  4997.7     .05       0  5001.7     .07       0
Bank Sta=4997.7,5001.7
XS Rating Curve= 0 ,0
Exp/Cntr=0.3,0.1

Type RM Length L Ch R = 1 ,44885   ,468,468,468
BEGIN DESCRIPTION:
North Creek 91.0
END DESCRIPTION:
XS GIS Cut Line= 3
      1991674.97     13939824.96        1991425.       13939525.
      1991324.97     13939474.99
#Sta/Elev= 30
  4609.3 1885.77  4647.4 1880.12  4666.9 1875.52  4671.2 1873.74  4678.6 1872.55
  4709.9 1863.03  4748.9 1849.11  4754.3 1848.48  4760.6 1845.43  4786.2 1838.42
  4802.9 1835.21  4839.5 1831.22  4845.9  1828.7  4858.3 1826.08  4867.2 1823.13
  4894.9 1820.96  4932.5 1820.47  4940.3 1820.96  4973.7 1819.77  4980.1 1819.21
  4988.3 1816.59  4988.6 1816.09  4992.3 1816.59  5001.4 1816.71  5014.9 1821.56
    5040 1840.06  5056.7 1849.65  5061.8 1853.72  5080.2 1863.95  5111.6 1875.16
#Mann= 3 ,-1 , 0
  4609.3     .07       0  4988.3     .05       0  4992.3     .07       0
Bank Sta=4988.3,4992.3
XS Rating Curve= 0 ,0
Exp/Cntr=0.3,0.1

Type RM Length L Ch R = 1 ,44417   ,458,458,458
BEGIN DESCRIPTION:
North Creek 90.0
END DESCRIPTION:
XS GIS Cut Line= 3
        1991825.       13939275.        1991775.       13939225.
      1991475.04     13939125.01
#Sta/Elev= 30
  4925.9 1840.72  4940.2 1838.79  4973.9 1831.65    4989  1826.1  4995.1  1824.5
  4998.7 1822.55  5001.8 1820.05    5005 1814.34  5009.3 1809.16  5009.6 1808.66
  5013.1 1808.66  5013.3 1809.16  5020.8 1809.78  5030.3 1812.82  5036.6 1813.53
  5065.1 1812.69  5079.8  1813.4    5083 1812.66  5094.8 1812.44  5128.2 1812.69
  5156.8 1812.41    5185 1813.37  5213.7 1815.26  5229.5 1817.81  5234.8 1819.12
  5244.3  1822.9  5260.9 1830.81  5264.3  1833.4  5282.2 1841.96  5312.8 1854.87
#Mann= 4 ,-1 , 0
  4925.9      .1       0  5009.3     .05       0  5013.3      .1       0
  5128.2     .07       0
Bank Sta=5009.3,5013.3
XS Rating Curve= 0 ,0
Exp/Cntr=0.3,0.1

Type RM Length L Ch R = 1 ,43959   ,610,610,610
BEGIN DESCRIPTION:
North Creek 89.0
END DESCRIPTION:
XS GIS Cut Line= 3
      1992074.96     13938974.98        1991775.       13938825.
      1991475.01       13938875.
#Sta/Elev= 30
  4669.2 1888.55  4681.4  1885.4  4718.5 1873.55  4740.9 1868.66  4764.4 1860.45
  4798.8  1848.3  4819.2 1844.39  4839.3 1838.43  4869.2 1823.74  4900.1 1810.54
  4912.8 1807.77  4924.3 1806.53  4947.2 1805.94  4983.3 1806.18  5013.7 1802.46
  5013.9 1801.96  5017.7 1802.46  5018.7 1803.51  5026.8 1806.19  5034.1 1809.78
  5096.1 1815.46  5103.9 1817.02  5125.2 1819.11  5166.9 1820.99  5205.9 1824.81
  5216.4 1826.94  5230.5 1831.76  5252.9  1838.9  5295.5 1856.83  5308.7 1861.45
#Mann= 7 ,-1 , 0
  4669.2     .07       0  4764.4      .1       0  4947.2     .07       0
  5013.7     .05       0  5017.7     .07       0  5166.9    .035       0
  5230.5     .07       0
Bank Sta=5013.7,5017.7
XS Rating Curve= 0 ,0
Exp/Cntr=0.3,0.1

Type RM Length L Ch R = 1 ,43349   ,193,193,193
BEGIN DESCRIPTION:
North Creek 88.0
END DESCRIPTION:
XS GIS Cut Line= 3
        1992075.       13938675.      1991759.04     13938280.08
      1991474.98     13938124.99
#Sta/Elev= 30
    4466 1837.43  4488.3 1833.59    4511 1831.48  4596.4 1820.32  4651.6 1816.15
  4683.9 1814.82    4733 1809.41  4888.4 1798.58  4996.3 1797.63  5005.2 1796.83
  5021.5 1792.66  5025.6 1791.64  5025.8 1791.14  5029.6 1791.64    5031 1795.09
  5034.4 1798.72  5051.5  1801.3  5069.3 1810.62  5085.7 1811.99  5091.4 1814.27
  5109.1 1828.04  5114.4 1834.24  5122.4 1841.41    5132 1847.77  5157.7 1863.32
  5179.9 1874.43  5184.8 1878.25  5208.7 1885.44  5257.2 1902.97  5295.4  1912.6
#Mann= 7 ,-1 , 0
    4466      .1       0    4511     .07       0  4888.4    .035       0
  5021.5     .07       0  5025.6    .035       0  5029.6     .07       0
    5132      .1       0
Bank Sta=5025.6,5029.6
XS Rating Curve= 0 ,0
Exp/Cntr=0.3,0.1

Type RM Length L Ch R = 1 ,43156   ,603,603,603
BEGIN DESCRIPTION:
North Creek 87.0
END DESCRIPTION:
XS GIS Cut Line= 3
      1992326.37     13938575.76      1991884.46     13938157.56
      1991725.03     13937875.06
#Sta/Elev= 30
  4396.5 1867.83    4421 1864.08  4456.2 1853.88  4472.7  1847.2    4500 1841.96
  4542.9 1830.42  4589.2 1823.61  4599.8 1823.34  4699.6 1811.63  4751.6 1807.25
    4799 1800.97  4819.8 1800.23  4871.4 1795.51  4926.6 1792.62  4979.6 1794.54
  4982.9 1793.92  4988.1 1790.63  4999.4 1789.48  4999.6 1788.98  5003.4 1789.48
  5008.2 1790.28  5015.1 1794.21    5022 1800.76  5029.4  1805.6  5049.5 1822.92
  5062.4 1831.13  5170.3 1866.79  5218.2 1884.73  5266.5 1902.56  5329.3 1921.16
#Mann= 8 ,-1 , 0
  4396.5     .07       0    4421    .035       0  4699.6      .1       0
  4819.8     .07       0  4999.4     .05       0  5003.4     .07       0
  5029.4      .1       0  5218.2     .07       0
Bank Sta=4999.4,5003.4
XS Rating Curve= 0 ,0
Exp/Cntr=0.3,0.1

Type RM Length L Ch R = 1 ,42553   ,391,391,391
BEGIN DESCRIPTION:
North Creek 86.0
END DESCRIPTION:
XS GIS Cut Line= 3
      1992618.27     13938074.28        1992275.       13937925.
      1991974.96     13937824.99
#Sta/Elev= 30
  4625.7 1832.28  4652.9 1827.34  4670.7 1826.01  4700.1  1821.1  4709.9  1820.8
  4726.3  1817.9    4776 1815.08  4788.4 1813.42  4837.5 1810.26  4929.1 1800.28
  4942.2 1795.54  4950.6 1789.69  4958.5 1785.97  4981.4 1779.11  4989.3 1778.48
  4989.5 1777.98  4993.3 1778.48  4997.8 1781.16    5001 1784.71  5004.1 1785.46
  5042.1 1786.55  5136.9  1785.3  5165.4 1786.23  5187.6 1792.25  5222.3 1806.23
  5250.2 1818.94  5274.6 1830.89  5276.9 1832.85  5295.1 1840.96  5316.3  1851.7
#Mann= 4 ,-1 , 0
  4625.7     .07       0  4989.3     .05       0  4993.3     .07       0
  5250.2      .1       0
Bank Sta=4989.3,4993.3
XS Rating Curve= 0 ,0
Exp/Cntr=0.3,0.1

Type RM Length L Ch R = 1 ,42162   ,515,515,515
BEGIN DESCRIPTION:
North Creek 85.0
END DESCRIPTION:
XS GIS Cut Line= 3
      1992642.86     13938022.43      1992272.22     13937555.96
        1992225.       13937275.
#Sta/Elev= 30
    4419 1827.62  4482.7 1816.91  4566.3 1808.95  4706.9 1799.44  4740.5 1795.77
  4766.2 1790.18  4789.9  1787.6  4845.7 1781.78    4954 1782.22  4987.8  1780.6
  4997.2 1778.99  5002.2 1775.53  5035.7 1772.65    5036 1772.15  5039.7 1772.65
  5049.5 1778.99  5076.8 1781.37  5095.3 1789.02  5108.1 1797.23  5119.5 1802.02
  5134.7 1812.12  5140.8 1819.08  5147.1 1823.76    5159 1837.03  5173.2 1845.45
  5219.9 1866.17  5247.3 1887.38  5259.4 1895.18  5283.8 1906.88  5299.7 1912.43
#Mann= 6 ,-1 , 0
    4419     .07       0  4566.3      .1       0  4766.2     .07       0
  4789.9      .1       0  5035.7     .05       0  5039.7      .1       0
Bank Sta=5035.7,5039.7
XS Rating Curve= 0 ,0
Exp/Cntr=0.3,0.1

Type RM Length L Ch R = 1 ,41647   ,469,469,469
BEGIN DESCRIPTION:
North Creek 84.0
END DESCRIPTION:
XS GIS Cut Line= 3
       1992882.9     13937853.58        1992675.       13937525.
      1992275.03     13937175.03
#Sta/Elev= 30
  4606.7 1821.07  4638.4 1812.26  4694.9 1812.82  4708.4 1810.43  4768.7 1803.49
  4850.3 1790.74  4868.1 1790.03  4924.9 1779.48  4949.3 1778.73  4973.1 1775.12
  4984.1 1772.38  5003.6    1763  5003.9  1762.5  5007.6    1763  5024.8 1769.06
  5065.9 1768.82  5109.8 1774.23  5169.5 1775.91  5191.9 1779.21  5205.4 1784.11
  5233.3 1799.08  5292.1 1825.48  5326.7 1846.52  5352.2 1859.28  5369.5 1865.92
  5384.1 1874.53  5415.1 1896.89  5436.6 1907.17  5488.2 1925.49    5527 1933.96
#Mann= 5 ,-1 , 0
  4606.7    .035       0  4708.4     .07       0  4973.1      .1       0
  5003.6     .05       0  5007.6      .1       0
Bank Sta=5003.6,5007.6
XS Rating Curve= 0 ,0
Exp/Cntr=0.3,0.1

Type RM Length L Ch R = 1 ,41178   ,454,454,454
BEGIN DESCRIPTION:
North Creek 83.0
END DESCRIPTION:
XS GIS Cut Line= 3
        1993175.       13937425.        1992925.       13937175.
      1992575.02     13936875.02
#Sta/Elev= 30
  4646.7 1802.46  4680.8 1800.51  4703.2  1794.4  4715.9 1794.99  4741.4 1791.49
  4775.3  1784.2  4784.8 1780.19  4801.7 1775.94  4816.6 1773.84  4977.8  1766.7
    4990 1764.88  5001.1 1759.81  5001.3 1758.42  5001.5 1757.92  5005.3 1758.42
  5027.3 1759.95  5043.7 1761.55  5058.6 1766.94  5117.1 1769.93  5167.1 1775.58
  5196.9 1782.79  5201.7 1785.51  5243.7 1798.66  5275.6 1815.59  5320.2 1847.79
  5351.9 1864.51    5370 1876.25  5407.5 1896.33  5428.8 1906.07  5461.2 1915.84
#Mann= 7 ,-1 , 0
  4646.7    .035       0    4990     .07       0  5001.3     .05       0
  5005.3     .07       0  5027.3    .035       0  5117.1      .1       0
    5370    .035       0
Bank Sta=5001.3,5005.3
XS Rating Curve= 0 ,0
Exp/Cntr=0.3,0.1

Type RM Length L Ch R = 1 ,40724   ,466,466,466
BEGIN DESCRIPTION:
North Creek 82.0
END DESCRIPTION:
XS GIS Cut Line= 3
        1993275.       13936925.        1993075.       13936775.
      1992675.01       13936725.
#Sta/Elev= 30
  4750.5  1780.1  4767.1 1780.32  4775.7 1778.29  4786.7 1771.29  4790.7 1765.86
  4794.2  1759.1  4816.7 1759.52  4854.2 1757.67  4857.1 1761.82  4861.7 1764.06
  4880.4 1762.82  4906.7 1763.81  4947.9 1761.85  4977.9 1762.38  4996.7 1759.65
  5003.4 1754.23  5004.5 1751.77  5004.8 1751.27  5008.6 1751.77  5031.9 1754.92
    5041 1754.85  5060.9 1757.69  5079.1 1757.87  5118.4 1766.95  5136.5 1776.54
    5170 1804.62  5186.5 1813.52  5239.3 1833.97  5328.8 1871.07  5403.6 1899.86
#Mann= 6 ,-1 , 0
  4750.5    .035       0  5004.5    .035       0  5008.6    .035       0
  5031.9     .07       0  5186.5      .1       0  5328.8     .07       0
Bank Sta=5004.5,5008.6
XS Rating Curve= 0 ,0
Exp/Cntr=0.3,0.1

Type RM Length L Ch R = 1 ,40258   ,432,432,432
BEGIN DESCRIPTION:
North Creek 81.0
END DESCRIPTION:
XS GIS Cut Line= 4
      1993654.92     13936662.54        1993225.       13936425.
      1993170.59     13936405.36      1992825.04     13936524.99
#Sta/Elev= 30
  4515.3 1799.52  4574.6 1795.57  4590.1 1792.28  4644.2 1786.43  4672.5 1782.24
  4685.1 1781.16    4698 1777.83  4724.8 1777.99  4752.8 1771.21  4818.3 1771.66
  4872.7 1769.82  4900.2 1764.55  4937.9 1752.03  4991.7 1746.38  4992.1 1745.88
  4996.7 1746.38  5005.2 1747.54  5012.8 1746.77  5044.7 1750.73  5064.3 1755.45
  5082.2 1757.02    5140 1761.66  5197.2 1769.45  5241.6 1782.97  5273.4  1789.6
  5298.8 1797.59  5330.5 1803.12  5346.4 1808.27  5384.5 1814.76    5430  1826.1
#Mann= 7 ,-1 , 0
  4515.3     .07       0  4644.2    .035       0  4672.5    .063       0
  4818.3    .035       0  4991.7    .035       0  4996.7    .035       0
  5082.2     .07       0
Bank Sta=4991.7,4996.7
XS Rating Curve= 0 ,0
Exp/Cntr=0.3,0.1

Type RM Length L Ch R = 1 ,39826   ,455,455,455
BEGIN DESCRIPTION:
North Creek 80.0
END DESCRIPTION:
XS GIS Cut Line= 3
      1993524.96     13936124.98        1993425.       13936075.
      1993024.97     13935774.98
#Sta/Elev= 30
  4888.6 1766.29  4909.6 1765.43  4935.5  1760.5  4955.6 1760.13    4969 1758.35
  4981.2 1751.77  4989.1 1744.19  4999.2 1740.06  5000.8 1740.05  5001.2 1739.55
  5005.9 1740.05  5017.8 1742.68    5027 1743.75  5047.8 1743.08  5055.3 1743.75
  5074.1 1751.45  5081.6 1752.19    5151 1751.68  5179.1 1751.04  5231.6 1753.52
  5273.4 1754.42  5307.7 1757.42  5314.1 1759.17    5342 1763.53  5361.3  1769.6
  5392.8 1783.16    5417 1796.17  5434.2 1807.86  5459.2 1820.49  5500.4 1830.25
#Mann= 4 ,-1 , 0
  4888.6    .035       0  5000.8    .035       0  5005.9    .035       0
    5151     .07       0
Bank Sta=5000.8,5005.9
XS Rating Curve= 0 ,0
Exp/Cntr=0.3,0.1

Type RM Length L Ch R = 1 ,39371   ,431,431,431
BEGIN DESCRIPTION:
North Creek 79.0
END DESCRIPTION:
XS GIS Cut Line= 3
      1994039.12     13935703.72        1993425.       13935675.
        1993025.       13935725.
#Sta/Elev= 30
  4390.1  1830.9  4415.2 1819.51  4466.3 1806.07  4505.9 1790.85  4554.7 1775.75
  4571.9 1772.09  4661.6 1763.06  4697.5  1763.2  4726.8 1759.62  4760.6 1761.06
  4808.6 1758.46  4832.7 1754.13  4856.7 1752.87  4936.3  1739.4  4958.8 1740.01
  4970.8 1736.75  4995.1 1736.01  4995.5 1735.51  5000.6 1736.01  5012.9 1743.67
    5022 1746.77  5085.8 1747.51  5167.1 1750.23  5206.4 1758.52    5254 1779.19
  5309.2 1789.37  5336.4 1798.28  5354.5  1806.4  5357.6 1817.68    5408 1831.38
#Mann= 5 ,-1 , 0
  4390.1      .1       0  4661.6    .035       0  4995.1    .035       0
  5000.6    .035       0  5085.8     .07       0
Bank Sta=4995.1,5000.6
XS Rating Curve= 0 ,0
Exp/Cntr=0.3,0.1

Type RM Length L Ch R = 1 ,38940   ,446,446,446
BEGIN DESCRIPTION:
North Creek 78.0
END DESCRIPTION:
XS GIS Cut Line= 3
      1993925.01       13935275.        1993525.       13935275.
      1993125.02       13935375.
#Sta/Elev= 30
  4594.6 1805.89    4640  1790.7  4685.9 1777.49  4712.6 1767.33  4730.9 1768.56
  4766.2 1755.96  4775.6 1753.49  4812.6 1752.98  4844.6 1751.17  4865.6 1745.99
  4955.9 1736.49    5010  1733.9  5013.5 1731.32  5013.9 1730.82    5019 1731.32
  5056.4 1733.41  5078.4 1741.64  5092.4 1743.14  5251.6 1745.87  5291.4 1762.42
    5315 1765.85  5316.6 1767.31  5319.3  1773.7  5322.4 1776.56  5327.4 1776.41
  5337.8 1781.96    5378 1783.67  5382.5 1788.68  5384.2 1793.25  5406.9 1797.74
#Mann= 6 ,-1 , 0
  4594.6     .07       0    4640    .035       0  4766.2    .063       0
  4812.6    .035       0  5013.5    .035       0    5019    .035       0
Bank Sta=5013.5,5019
XS Rating Curve= 0 ,0
Exp/Cntr=0.3,0.1

Type RM Length L Ch R = 1 ,38494   ,482,482,482
BEGIN DESCRIPTION:
North Creek 77.0
END DESCRIPTION:
XS GIS Cut Line= 3
      1993975.03     13934724.99        1993575.       13934875.
      1993175.03     13935024.99
#Sta/Elev= 30
  4572.4 1816.51  4591.5 1812.13  4610.2 1809.92  4634.3 1803.93  4646.1 1798.19
  4661.6 1796.35  4674.9 1793.33  4694.2 1780.29  4713.4 1772.99  4726.2 1770.72
  4758.2 1761.71  4783.9 1763.06  4835.1 1743.24  4894.1 1742.04  4905.6 1740.26
  4921.6 1733.82  4950.4 1731.08  4973.3 1725.85  4973.8 1725.35  4978.9 1725.85
  5004.9 1729.51  5030.6  1736.5    5083  1736.8  5126.7 1735.45  5136.9  1736.9
  5210.5 1737.35  5280.5  1740.6  5349.9 1755.75  5373.5  1760.2  5426.8 1767.29
#Mann= 8 ,-1 , 0
  4572.4     .07       0  4661.6    .035       0  4973.3    .035       0
  4978.9    .035       0    5083     .07       0  5210.5    .035       0
  5349.9     .07       0  5373.5    .035       0
#XS Ineff= 2 , 0
                         5047.35         1738.56
Permanent Ineff=
       F       F
Bank Sta=4973.3,4978.9
XS Rating Curve= 0 ,0
Exp/Cntr=0.3,0.1

Type RM Length L Ch R = 1 ,38012   ,466,466,466
BEGIN DESCRIPTION:
North Creek 76.0
END DESCRIPTION:
XS GIS Cut Line= 3
      1993874.96     13934524.99        1993475.       13934425.
        1993175.       13934525.
#Sta/Elev= 30
  4587.3 1805.03  4598.6 1804.52  4607.8  1799.1  4631.2 1792.15  4641.9 1785.53
  4669.7 1772.21  4682.1 1763.96  4694.4 1753.89    4705 1751.98  4719.2 1751.96
  4727.7 1748.17  4737.7 1741.21  4754.9 1734.66    4781 1733.75  4793.4 1736.29
  4808.8 1737.51    4849 1738.49  4961.7 1723.83  4988.4 1721.76  4988.9 1721.26
  4994.1 1721.76  5005.6 1723.77  5063.8 1725.39  5155.5  1731.5    5165 1733.49
  5228.3 1740.63  5244.1 1744.01  5274.7 1746.72  5275.2 1746.76  5315.8 1751.68
#Mann= 6 ,-1 , 0
  4587.3    .035       0  4961.7     .07       0  4988.4     .05       0
  4994.1     .07       0  5274.7    .035       0  5275.2     .07       0
Bank Sta=4988.4,4994.1
XS Rating Curve= 0 ,0
Exp/Cntr=0.3,0.1

Type RM Length L Ch R = 1 ,37546   ,466,466,466
BEGIN DESCRIPTION:
North Creek 75.0
END DESCRIPTION:
XS GIS Cut Line= 3
        1993925.       13934125.        1993525.       13933975.
        1993175.       13934075.
#Sta/Elev= 30
  4572.9 1810.81    4606 1800.62  4628.4 1798.03  4645.6 1792.19  4660.4 1781.71
  4675.6 1775.51  4724.7 1770.12  4746.9 1760.06    4763 1747.84    4775 1746.24
    4795 1746.83  4818.7 1739.73  4833.4 1732.38    4867 1734.99  4910.3 1735.23
  4938.9 1726.02  4958.4 1724.79  4973.9  1721.2  4996.9    1720  5006.3 1712.57
  5012.8 1712.36  5013.3 1711.86  5018.5 1712.36  5021.9 1715.03  5043.7 1722.91
  5090.5  1720.4  5168.5 1719.38  5224.7 1722.88  5296.5 1734.05  5364.1 1739.22
#Mann= 6 ,-1 , 0
  4572.9     .07       0  4645.6    .035       0    4775    .063       0
    4867    .035       0  5012.8    .035       0  5018.5    .035       0
Bank Sta=5012.8,5018.5
XS Rating Curve= 0 ,0
Exp/Cntr=0.3,0.1

Type RM Length L Ch R = 1 ,37080   ,630,630,630
BEGIN DESCRIPTION:
North Creek 74.0
END DESCRIPTION:
XS GIS Cut Line= 4
       1993781.2     13933573.98        1993575.       13933525.
      1993497.57     13933518.47      1993225.05     13933674.97
#Sta/Elev= 30
  4783.2  1763.8    4809  1739.9  4818.3 1733.27  4821.4 1732.22  4827.5 1730.91
  4883.9 1733.43  4895.4 1733.31  4916.9 1736.91  4929.3 1736.76  4941.6 1734.95
  4953.2 1731.83  4964.4 1726.86  4969.3 1722.83  4981.7 1717.38  5000.1 1706.34
  5005.3 1705.05  5012.1 1706.01  5018.3 1704.69  5018.8 1704.19    5024 1704.69
  5024.7 1706.81  5030.2  1712.6  5033.2 1713.25  5071.9 1711.22  5175.9 1712.55
  5234.9 1714.85  5307.5 1715.33  5324.8 1716.46    5349 1723.77  5387.1 1724.23
#Mann= 4 ,-1 , 0
  4783.2    .063       0  4883.9    .035       0  5018.3    .035       0
    5024    .035       0
#XS Ineff= 2 , 0
                         5035.66         1713.13
Permanent Ineff=
       F       F
Bank Sta=5018.3,5024
XS Rating Curve= 0 ,0
Exp/Cntr=0.3,0.1

Type RM Length L Ch R = 1 ,36450   ,297,297,297
BEGIN DESCRIPTION:
North Creek 73.0
END DESCRIPTION:
XS GIS Cut Line= 3
      1994162.21     13932936.82       1993577.8     13932954.89
      1993225.08     13933024.98
#Sta/Elev= 30
  4412.7 1740.59  4484.6 1731.54  4506.7 1727.88  4526.7 1728.89  4584.9 1721.67
  4617.9 1727.37    4675 1729.51  4689.4 1727.33  4699.7 1721.57    4708 1718.51
    4774 1715.46    4828 1704.77    4831 1708.43    4835 1709.37  4900.1 1704.14
  4951.1 1706.06  4954.1 1705.61  4963.1 1697.59  4976.5  1692.7    4977  1692.2
  4985.7  1692.7  4996.1  1697.7  4999.1 1703.66  5005.3 1705.59  5029.7 1703.82
  5103.4 1705.12  5283.6  1716.2  5320.3  1722.5  5344.8 1723.69    5357 1726.83
#Mann= 7 ,-1 , 0
  4412.7     .07       0  4484.6    .035       0  4526.7    .063       0
  4699.7    .035       0  4976.5    .035       0  4985.7    .035       0
  5103.4     .07       0
#XS Ineff= 2 , 0
         4833.57 1709.88
Permanent Ineff=
       F       F
Bank Sta=4976.5,4985.7
XS Rating Curve= 0 ,0
Exp/Cntr=0.3,0.1

Type RM Length L Ch R = 1 ,36153   ,473,473,473
BEGIN DESCRIPTION:
North Creek 72.0
END DESCRIPTION:
XS GIS Cut Line= 3
      1993724.99       13932675.        1993525.       13932675.
        1993125.       13932525.
#Sta/Elev= 30
    4800 1706.48  4828.9 1705.89  4849.9 1703.36  4876.9 1701.86  4885.9 1703.24
    4897 1703.65    4927 1701.74  4948.9 1701.85    4963 1700.46  4981.9 1700.76
  4990.9 1695.79  4999.9 1692.11  5008.6 1690.63  5009.1 1690.13  5017.8 1690.63
  5022.5 1693.79  5041.6 1701.45  5048.1 1702.49  5059.5 1701.95  5131.3 1699.74
    5205 1699.47    5237 1700.91  5265.8 1706.04  5278.7 1706.17  5294.7 1711.26
  5320.3 1723.44  5339.4 1734.19  5384.4 1753.05  5416.3 1770.38  5427.2 1774.55
#Mann= 4 ,-1 , 0
    4800     .07       0  5008.6     .05       0  5017.8     .07       0
  5059.5    .035       0
#XS Ineff= 2 , 0
                         5053.85         1701.76
Permanent Ineff=
       F       F
Bank Sta=5008.6,5017.8
XS Rating Curve= 0 ,0
Exp/Cntr=0.3,0.1

Type RM Length L Ch R = 1 ,35680   ,440,440,440
BEGIN DESCRIPTION:
North Creek 71.0
END DESCRIPTION:
XS GIS Cut Line= 3
      1993835.77     13932307.62       1993376.5     13932249.97
      1993175.01       13932225.
#Sta/Elev= 30
  4535.2  1706.1  4574.9 1706.26  4627.6 1702.96    4673 1703.07  4694.3 1701.25
  4725.4 1699.34  4760.6 1700.18  4768.4 1699.49  4781.8 1695.46  4793.2 1695.01
  4846.3  1698.5  4892.2 1697.31    4939 1693.98  4954.1 1690.15  4979.8 1687.03
  4980.3 1686.53    4989 1687.03  4990.4  1689.9  5023.6 1706.99  5042.4 1715.14
    5069 1731.36  5082.8 1736.27  5090.1 1741.89  5096.2 1746.94  5111.3 1754.45
  5132.5  1762.8  5147.6 1771.33  5156.7 1773.34  5171.8 1786.38  5201.1 1800.34
#Mann= 7 ,-1 , 0
  4535.2    .035       0  4694.3     .07       0  4793.2    .035       0
  4892.2     .07       0  4979.8     .05       0    4989     .07       0
  5090.1    .035       0
Bank Sta=4979.8,4989
XS Rating Curve= 0 ,0
Exp/Cntr=0.3,0.1

Type RM Length L Ch R = 1 ,35240   ,448,448,448
BEGIN DESCRIPTION:
North Creek 70.0
END DESCRIPTION:
XS GIS Cut Line= 3
      1993725.04     13931975.03        1993575.       13931875.
      1993175.04       13931925.
#Sta/Elev= 30
  4819.7 1697.55    4833 1697.08  4882.5  1696.1  4899.8 1692.94  4908.6 1692.58
    4923 1689.04  4937.4 1686.96  4951.9 1687.04  4980.7 1681.46  4990.1  1681.4
  4990.6  1680.9  4999.4  1681.4  5029.2 1686.19  5036.5  1689.2  5043.8 1692.53
  5050.3 1694.21  5059.4 1693.58  5083.6 1700.33  5107.8  1709.4  5123.2 1717.97
    5141 1722.35  5183.4  1738.3  5199.3 1742.61  5230.1 1753.57    5271 1763.37
  5292.2 1769.83  5310.3 1777.16  5361.7 1790.36  5373.8 1796.62  5403.1 1809.17
#Mann= 5 ,-1 , 0
  4819.7    .035       0    4833     .07       0  4990.1     .05       0
  4999.4     .07       0  5036.5    .035       0
Bank Sta=4990.1,4999.4
XS Rating Curve= 0 ,0
Exp/Cntr=0.3,0.1

Type RM Length L Ch R = 1 ,34792   ,468,468,468
BEGIN DESCRIPTION:
North Creek 69.0
END DESCRIPTION:
XS GIS Cut Line= 3
      1994108.65     13931785.24        1993725.       13931475.
      1993251.13     13931243.69
#Sta/Elev= 30
  4511.4 1707.09  4665.4 1700.63  4717.9 1697.62  4737.2 1692.56  4760.3 1695.16
  4802.8 1691.66  4845.2 1691.67  4924.4 1688.62  4937.8 1686.57    4952  1680.9
  4971.4 1678.27  4977.3 1675.64  4977.8 1675.14  4986.7 1675.64  5020.3 1681.95
    5047 1684.08    5077 1691.42  5117.1 1693.25  5155.8  1699.8  5190.2 1703.02
  5227.3 1703.56    5259 1708.97    5284 1716.69  5310.6 1719.96  5344.1 1730.16
  5360.8 1735.43  5402.6 1743.52  5454.3 1756.94  5512.5 1760.26  5532.1  1764.3
#Mann= 7 ,-1 , 0
  4511.4     .07       0  4665.4    .035       0    4952     .07       0
  4977.3     .05       0  4986.7     .07       0  5190.2    .035       0
  5344.1     .07       0
Bank Sta=4977.3,4986.7
XS Rating Curve= 0 ,0
Exp/Cntr=0.3,0.1

Type RM Length L Ch R = 1 ,34324   ,513,513,513
BEGIN DESCRIPTION:
North Creek 68.0
END DESCRIPTION:
XS GIS Cut Line= 3
      1994389.22     13931490.08        1993925.       13931075.
      1993540.45     13930938.17
#Sta/Elev= 30
  4381.8 1713.88  4515.5 1703.27  4556.1 1701.98  4695.7 1689.06  4728.1 1684.31
  4822.2 1685.94  4891.2 1686.31  4931.6 1684.24  4944.3 1681.64  4965.5 1672.79
  4977.8 1670.67  4978.3 1670.17  4987.4 1670.67  4991.1 1673.44  5013.1 1675.75
    5029 1679.91  5037.3 1681.03  5053.3 1679.69  5075.6 1689.28  5097.8 1691.74
  5120.3 1691.64  5223.8 1697.15  5271.5 1700.25    5295 1704.77  5301.6 1703.49
  5323.1 1711.49  5331.9 1712.81    5359 1718.58  5397.2 1721.28  5412.7 1725.82
#Mann= 8 ,-1 , 0
  4381.8    .035       0  4822.2     .07       0  4977.8     .05       0
  4987.4     .07       0  5120.3    .035       0  5223.8     .07       0
  5271.5    .035       0  5331.9     .07       0
Bank Sta=4977.8,4987.4
XS Rating Curve= 0 ,0
Exp/Cntr=0.3,0.1

Type RM Length L Ch R = 1 ,33811   ,437,437,437
BEGIN DESCRIPTION:
North Creek 67.0
END DESCRIPTION:
XS GIS Cut Line= 4
      1994505.33     13931133.44      1994365.76     13930942.03
      1994068.97       13930632.      1993689.16      13930593.8
#Sta/Elev= 30
  4758.3  1713.4  4813.4 1707.59    4869 1699.67  4892.7  1693.7    4939 1677.45
  4986.6 1667.16  4987.1 1666.66  4996.3 1667.16  5004.2 1667.59  5029.7 1669.56
  5045.2 1678.92  5056.9 1682.63  5111.6 1682.38  5119.9 1683.32  5143.7 1681.45
  5187.1 1680.97  5237.8 1684.75  5275.8 1685.33  5286.8 1684.51  5341.6 1684.42
  5360.6 1685.25  5408.3 1683.41  5421.3 1684.58  5473.5 1683.54  5585.1 1685.06
  5711.7 1692.89    5763 1697.55    5775 1699.82  5790.1 1700.49  5806.1 1703.89
#Mann= 6 ,-1 , 0
  4758.3     .07       0    4939      .1       0  4986.6     .05       0
  4996.3      .1       0  5004.2     .07       0  5237.8    .035       0
Bank Sta=4986.6,4996.3
XS Rating Curve= 0 ,0
Exp/Cntr=0.3,0.1

Type RM Length L Ch R = 1 ,33374   ,464,464,464
BEGIN DESCRIPTION:
North Creek 66.0
END DESCRIPTION:
XS GIS Cut Line= 3
      1994816.72      13930533.2        1994425.       13930525.
       1993970.7      13930511.9
#Sta/Elev= 30
  4608.2 1725.44  4642.9 1723.96  4678.9 1715.67  4705.8 1713.54  4723.9 1710.33
  4744.9 1708.61  4804.4 1700.75  4840.9 1696.91  4891.9 1694.81  4915.9  1692.7
  4926.5 1685.26  4947.1 1673.66  4966.9 1664.47  4981.9 1662.32  4986.1 1659.97
  4986.6 1659.47  4995.8 1659.97  4996.9  1662.3  5001.5 1663.27  5008.8 1664.42
  5038.9 1674.52    5051 1677.54  5058.6 1678.18    5081 1675.96    5114  1675.5
    5141 1676.38  5169.2 1679.85    5204 1680.96    5222 1682.66  5454.5 1683.05
#Mann= 6 ,-1 , 0
  4608.2    .035       0  4705.8     .07       0  4804.4      .1       0
  4986.1     .05       0  4995.8      .1       0  5001.5    .035       0
Bank Sta=4986.1,4995.8
XS Rating Curve= 0 ,0
Exp/Cntr=0.3,0.1

Type RM Length L Ch R = 1 ,32910   ,460,460,460
BEGIN DESCRIPTION:
North Creek 65.0
END DESCRIPTION:
XS GIS Cut Line= 3
      1994474.96       13930075.        1994375.       13930075.
      1994175.06     13930174.97
#Sta/Elev= 30
  4895.3 1683.56  4912.2  1679.7  4924.2 1678.16  4932.5 1676.63  4939.2 1674.31
  4942.2 1672.55  4954.2 1668.06  4963.2  1663.7  4969.2  1661.8  4978.2 1659.88
  4991.4 1659.75  4991.9 1659.25  5000.7 1659.25  5001.2 1659.75  5001.8 1660.01
  5016.4 1660.11  5024.3 1660.96  5028.6 1661.99    5036 1664.64    5050 1668.86
  5056.7 1670.19    5060 1671.49  5063.4 1672.17  5070.1 1671.43  5086.8 1670.85
  5130.1 1671.58  5140.5 1672.12  5174.1 1676.05  5187.5 1677.08  5218.8 1678.12
#Mann= 5 ,-1 , 0
  4895.3      .1       0  4932.5     .07       0  4991.4     .05       0
  5001.2     .07       0    5036    .035       0
Bank Sta=4991.4,5001.2
XS Rating Curve= 0 ,0
Exp/Cntr=0.3,0.1

Type RM Length L Ch R = 1 ,32450   ,451,451,451
BEGIN DESCRIPTION:
North Creek 64.0
END DESCRIPTION:
XS GIS Cut Line= 3
      1994580.04     13929604.46        1994275.       13929675.
      1993902.77     13929844.02
#Sta/Elev= 30
  4686.9 1679.57  4701.2  1678.9  4818.4 1678.97  4879.8 1676.73  4895.2 1676.95
  4907.5 1678.32  4913.7 1678.43  4932.2 1675.98  4946.6 1675.23  4950.6 1674.36
    4963  1667.7    4966 1664.71  4972.2 1660.05  4985.9 1658.67  4986.4 1658.17
  4995.2 1658.17  4995.7 1658.67  5032.9 1659.19  5039.4 1659.76  5047.4 1661.39
  5065.8 1664.34    5102 1667.77  5111.9 1671.48  5115.2 1671.78  5138.3  1670.3
  5184.4 1673.16  5276.7 1677.36  5326.1 1678.04  5356.2 1677.76  5408.8 1679.73
#Mann= 5 ,-1 , 0
  4686.9     .07       0  4985.9     .05       0  4995.7     .07       0
  5047.4    .035       0  5356.2     .07       0
Bank Sta=4985.9,4995.7
XS Rating Curve= 0 ,0
Exp/Cntr=0.3,0.1

Type RM Length L Ch R = 1 ,31999   ,465,465,465
BEGIN DESCRIPTION:
North Creek 63.0
END DESCRIPTION:
XS GIS Cut Line= 5
      1994801.21     13929399.14      1994477.61     13929271.07
        1994225.       13929275.      1994042.23     13929307.17
      1993855.99     13929829.95
#Sta/Elev= 30
  4403.9  1681.5  4445.8 1680.75    4467 1678.94  4582.6 1675.35  4906.5 1671.72
  4939.5 1669.63  4951.5 1665.69  4969.5 1656.72  4982.5 1656.06    4983 1655.56
  4992.4 1656.06  5017.7 1657.11  5048.1 1656.61  5060.3 1658.99  5075.6 1659.23
  5109.1 1662.31  5143.8 1669.64  5163.9  1672.2  5190.1 1673.75  5207.6  1673.3
    5283 1675.09  5298.9 1673.98  5329.4 1674.05  5400.1 1676.34    5451 1676.25
  5463.8 1677.46  5479.6 1676.49  5505.2  1676.7  5667.6 1679.81  5745.1 1682.36
#Mann= 3 ,-1 , 0
  4403.9     .07       0  4982.5     .05       0  4992.4     .07       0
Bank Sta=4982.5,4992.4
XS Rating Curve= 0 ,0
Exp/Cntr=0.3,0.1

Type RM Length L Ch R = 1 ,31534   ,492,492,492
BEGIN DESCRIPTION:
North Creek 62.0
END DESCRIPTION:
XS GIS Cut Line= 4
      1994759.57     13929291.34      1994466.39     13928951.85
        1994175.       13928825.      1993830.55     13928662.78
#Sta/Elev= 30
  4237.4 1677.92  4384.4 1674.49  4435.8 1673.06  4519.7 1673.42  4601.3 1670.43
  4671.7 1669.66    4737 1666.48  4750.7 1660.88  4802.9 1659.71  4832.4 1659.85
  4892.1 1657.43  4912.6 1654.23  4926.5 1655.24  4976.4 1654.36  4985.4 1651.76
  4985.9 1651.26  4997.4 1651.76    5024 1661.66  5071.4 1675.35  5080.4 1676.71
  5093.9 1680.96  5114.2 1683.59  5123.4  1686.9  5141.3 1693.87  5172.8 1696.28
  5269.8 1696.56    5301 1702.14  5344.3 1705.94  5357.7 1705.97  5384.5 1711.32
#Mann= 8 ,-1 , 0
  4237.4     .07       0  4384.4    .035       0  4671.7     .07       0
  4802.9    .035       0  4926.5     .07       0  4985.4     .05       0
  4997.4     .07       0  5123.4    .035       0
Bank Sta=4985.4,4997.4
XS Rating Curve= 0 ,0
Exp/Cntr=0.3,0.1

Type RM Length L Ch R = 1 ,31042   ,423,423,423
BEGIN DESCRIPTION:
North Creek 61.0
END DESCRIPTION:
XS GIS Cut Line= 4
      1994963.99     13929144.92      1994723.66     13928627.94
        1994525.       13928475.      1993952.86     13928468.28
#Sta/Elev= 30
    4175 1680.52    4184 1679.76  4214.7 1678.66  4223.9  1676.9  4251.1 1677.18
  4381.3 1671.82  4396.8 1671.42  4436.4 1669.22  4489.3 1669.55  4589.7 1666.44
  4614.6  1667.1  4630.4  1665.6  4658.1 1666.79  4798.3  1663.7    4838  1663.1
  4879.6 1653.47  4902.3 1651.41  4998.7 1651.34  4999.2 1650.84  5010.8 1651.34
  5031.1 1653.76  5119.8 1657.66  5273.7 1666.26  5339.8 1669.25  5374.8 1672.27
  5452.8 1685.66  5471.3 1690.81  5516.2 1699.35  5536.8 1701.63    5568 1702.75
#Mann= 11 ,-1 , 0
    4175    .035       0    4184     .07       0  4381.3    .035       0
  4396.8     .07       0  4658.1    .035       0  4798.3      .1       0
  4998.7     .05       0  5010.8      .1       0  5119.8     .07       0
  5273.7    .035       0  5516.2     .07       0
Bank Sta=4998.7,5010.8
XS Rating Curve= 0 ,0
Exp/Cntr=0.3,0.1
