--- Palmer Creek.prj (project) ---

Proj Title=Palmer Creek Base Level Engineering
Current Plan=p01
Default Exp/Contr=0.3,0.1
English Units
Geom File=g01
Flow File=f01
Plan File=p01
BEGIN DESCRIPTION:
Palmer Creek
END DESCRIPTION:

--- Palmer Creek.p01 (plan) ---

Plan Title=Multiple Run
Short Identifier=Multiple
Geom File=g01
Flow File=f01
Subcritical Flow
K Sum by GR= 0
Std Step Tol= 0.01
Critical Tol= 0.01
Num of Std Step Trials= 20
Max Error Tol= 0.3
Flow Tol Ratio= 0.001
Split Flow NTrial= 30
Split Flow Tol= 0.02
Split Flow Ratio= 0.02
Log Output Level= 0
Friction Slope Method= 1
Unsteady Friction Slope Method= 2
Unsteady Bridges Friction Slope Method= 1
Parabolic Critical Depth
Global Vel Dist=  1 , 1 , 1
Global Log Level= 0
CheckData=True
Encroach Param= -1, 0, 0, 0
BEGIN DESCRIPTION:
Multiple Run
END DESCRIPTION:

--- Palmer Creek.f01 (steady flow) ---

Flow Title=Multiple
Number of Profiles=7
Profile Names=10-year,25-year,50-year,1pct_min,100-year,1pct_plu,500-year
River Rch & RM= Palmer Creek,Reach-1,37933
    3369    6035    8699    6045   12062   24066   22900
River Rch & RM= Palmer Creek,Reach-1,35226
    3521    6313    9107    6330   12631   25202   24001
River Rch & RM= Palmer Creek,Reach-1,33476
    4003    7237   10494    7328   14621   29173   28052
River Rch & RM= Palmer Creek,Reach-1,31301
    4187    7552   10931    7616   15196   30321   29026
River Rch & RM= Palmer Creek,Reach-1,24994
    4820    8692   12582    8761   17481   34878   33338
River Rch & RM= Palmer Creek,Reach-1,19546
    5962   10847   15787   11044   22035   43966   42432
River Rch & RM= Palmer Creek,Reach-1,10609
    6334   11540   16813   11770   23485   46859   45292
River Rch & RM= Palmer Creek,Reach-1,8891
    6667   12154   17716   12406   24752   49387   47759
River Rch & RM= Palmer Creek,Reach-1,2822
    6620   12052   17549   12275   24492   48868   47154
Boundary for River Rch & Prof#=Palmer Creek,Reach-1,1
Up Type=0
Dn Type=3
Dn Slope=0.005
Boundary for River Rch & Prof#=Palmer Creek,Reach-1,2
Up Type=0
Dn Type=3
Dn Slope=0.005
Boundary for River Rch & Prof#=Palmer Creek,Reach-1,3
Up Type=0
Dn Type=3
Dn Slope=0.005
Boundary for River Rch & Prof#=Palmer Creek,Reach-1,4
Up Type=0
Dn Type=3
Dn Slope=0.005
Boundary for River Rch & Prof#=Palmer Creek,Reach-1,5
Up Type=0
Dn Type=3
Dn Slope=0.005
Boundary for River Rch & Prof#=Palmer Creek,Reach-1,6
Up Type=0
Dn Type=3
Dn Slope=0.005
Boundary for River Rch & Prof#=Palmer Creek,Reach-1,7
Up Type=0
Dn Type=3
Dn Slope=0.005

--- Palmer Creek.g01 (geometry) ---

Geom Title=Existing Conditions

River Reach=Palmer Creek,Reach-1
Reach XY= 30
      1901975.00     13869425.00      1903043.27     13869025.18
      1904523.35     13869228.17      1904654.35     13869655.58
      1905615.87     13870268.26      1905432.09     13871075.00
      1905668.54     13871367.27      1907281.76     13870734.12
      1908168.26     13872015.87      1908804.82     13872225.30
      1909835.11     13871935.30      1910876.50     13873421.54
      1912181.19     13873132.81      1912785.50     13874234.82
      1913680.26     13874922.91      1914391.67     13874708.35
      1914725.00     13873982.07      1916176.50     13874871.39
      1916675.00     13874682.07      1917528.42     13875017.21
      1917930.11     13874130.11      1918367.05     13874078.00
      1918924.91     13876267.81      1921518.83     13873482.86
      1921969.12     13873326.96      1922314.87     13873964.68
      1922638.63     13873861.54      1923419.48     13872977.43
      1923730.16     13872080.41      1925275.00     13870825.00

Type RM Length L Ch R = 1,37933,470,470,470
BEGIN DESCRIPTION:
Palmer Creek 75.0
END DESCRIPTION:
XS GIS Cut Line= 3
      1902224.98     13869474.95      1902175.00     13869325.00
      1902074.99     13869124.98
#Sta/Elev= 30
  4837.4 1924.83  4848.2 1923.17  4869.0 1913.63  4890.1 1902.53  4911.1 1893.21
  4921.7 1883.95  4942.8 1873.47  4963.8 1860.62  4984.9 1851.58  5009.4 1852.08
  5028.9 1851.12  5029.4 1850.62  5034.7 1851.12  5048.6 1865.02  5062.5 1866.44
  5076.5 1869.79  5098.9 1879.45  5107.3 1884.63  5115.7 1891.18  5129.6 1906.22
  5152.0 1919.52  5160.4 1924.37  5166.0 1926.48  5174.4 1932.46  5182.7 1936.76
  5188.3 1938.01  5205.1 1945.86  5210.7 1946.92  5216.3 1950.52  5219.1 1950.52
#Mann=4,-1,0
  4837.4    0.07       0  4848.2     0.1       0  5028.9    0.05       0
  5034.7     0.1       0
Bank Sta=5028.9,5034.7
Exp/Cntr=0.3,0.1

Type RM Length L Ch R = 1,37463,481,481,481
BEGIN DESCRIPTION:
Palmer Creek 74.0
END DESCRIPTION:
XS GIS Cut Line= 3
      1902625.00     13869374.99      1902575.00     13869125.00
      1902524.99     13868974.96
#Sta/Elev= 30
  4744.6 1922.20  4747.1 1922.20  4765.0 1917.11  4816.0 1900.33  4826.2 1895.72
  4848.3 1880.94  4867.0 1871.01  4872.1 1870.60  4877.2 1863.45  4887.4 1859.24
  4918.0 1856.99  4928.2 1851.92  4938.4 1847.74  4966.0 1847.18  4966.5 1846.68
  4971.3 1846.68  4971.8 1847.18  4989.3 1847.40  5002.2 1848.21  5020.6 1857.43
  5041.7 1858.03  5052.2 1862.41  5073.3 1875.85  5083.9 1885.11  5094.4 1898.36
  5105.0 1903.50  5115.5 1910.61  5136.6 1916.45  5155.0 1923.77  5157.7 1923.77
#Mann=4,-1,0
  4744.6    0.07       0  4848.3     0.1       0  4966.0    0.05       0
  4971.8     0.1       0
Bank Sta=4966,4971.8
Exp/Cntr=0.3,0.1

Type RM Length L Ch R = 1,36982,559,559,559
BEGIN DESCRIPTION:
Palmer Creek 73.0
END DESCRIPTION:
XS GIS Cut Line= 3
      1903025.00     13869375.02      1903025.00     13869025.00
      1902975.01     13868875.04
#Sta/Elev= 30
  4654.5 1920.68  4664.5 1919.01  4674.5 1915.75  4714.5 1905.23  4744.5 1895.55
  4754.5 1891.36  4774.5 1887.50  4784.0 1884.30  4794.5 1880.98  4824.5 1873.79
  4844.5 1870.02  4894.5 1856.07  4944.5 1848.70  4951.6 1845.86  4952.1 1845.36
  4957.0 1845.36  4957.5 1845.86  5025.6 1846.55  5036.1 1848.77  5046.7 1852.24
  5057.2 1863.39  5067.8 1871.38  5099.4 1889.25  5109.9 1895.51  5120.5 1902.99
  5131.0 1908.09  5141.6 1915.23  5152.1 1921.40  5160.0 1925.72  5162.6 1925.72
#Mann=4,-1,0
  4654.5    0.07       0  4784.0     0.1       0  4951.6    0.05       0
  4957.5     0.1       0
Bank Sta=4951.6,4957.5
Exp/Cntr=0.3,0.1

Type RM Length L Ch R = 1,36423,327,327,327
BEGIN DESCRIPTION:
Palmer Creek 72.0
END DESCRIPTION:
XS GIS Cut Line= 3
      1903475.00     13869424.99      1903510.37     13869217.65
      1903607.40     13868875.78
#Sta/Elev= 30
  4797.6 1919.80  4817.9 1918.42  4830.2 1916.34  4838.2 1913.12  4858.5 1901.02
  4868.6 1893.12  4885.3 1875.86  4890.4 1876.21  4909.2 1865.37  4924.0 1859.20
  4939.6 1853.94  4945.5 1849.54  4970.0 1841.54  4996.5 1837.24  4997.0 1836.74
  5004.5 1837.24  5052.3 1838.51  5062.7 1841.50  5079.0 1850.74  5118.1 1853.98
  5145.8 1866.17  5152.0 1871.17  5157.2 1872.03  5186.0 1884.91  5191.1 1884.26
  5197.8 1888.45  5225.1 1898.38  5230.2 1897.86  5298.1 1920.06  5363.3 1931.99
#Mann=4,-1,0
  4797.6    0.07       0  4924.0     0.1       0  4996.5    0.05       0
  5004.5     0.1       0
Bank Sta=4996.5,5004.5
Exp/Cntr=0.3,0.1

Type RM Length L Ch R = 1,36096,463,463,463
BEGIN DESCRIPTION:
Palmer Creek 71.0
END DESCRIPTION:
XS GIS Cut Line= 3
      1903775.01     13869374.98      1903825.00     13869275.00
      1903675.00     13868874.99
#Sta/Elev= 30
  4879.4 1911.44  4893.4 1908.15  4901.7 1905.00  4910.1 1899.49  4914.4 1899.08
  4915.7 1898.95  4924.1 1886.14  4932.5 1870.37  4938.1 1867.77  4954.9 1853.36
  4960.4 1852.85  4968.8 1843.04  4977.2 1838.72  5051.3 1836.96  5051.8 1836.46
  5059.3 1836.96  5061.5 1838.68  5091.8 1842.26  5116.7 1849.43  5152.3 1850.72
  5226.1 1865.11  5262.6 1875.89  5311.6 1896.64  5317.8 1900.19  5348.1 1911.07
  5354.3 1914.89  5373.0 1921.63  5378.3 1922.27  5403.3 1930.03  5418.4 1932.92
#Mann=4,-1,0
  4879.4    0.07       0  4914.4     0.1       0  5051.3    0.05       0
  5059.3     0.1       0
Bank Sta=5051.3,5059.3
Exp/Cntr=0.3,0.1

Type RM Length L Ch R = 1,35633,407,407,407
BEGIN DESCRIPTION:
Palmer Creek 70.0
END DESCRIPTION:
XS GIS Cut Line= 3
      1904075.01     13869524.98      1904212.37     13869238.47
      1904275.00     13868825.02
#Sta/Elev= 30
  4668.2 1916.16  4704.9 1911.24  4722.0 1905.25  4772.9 1893.26  4780.8 1889.97
  4812.3 1881.71  4818.2 1877.72  4846.4 1869.74  4908.8 1856.25  4914.4 1854.13
  4923.2 1838.96  4931.5 1837.43  5005.6 1837.17  5006.1 1836.67  5013.7 1837.17
  5019.8 1837.18  5029.9 1840.55  5035.9 1845.02  5060.2 1852.10  5080.5 1850.23
  5131.0 1849.34  5161.4 1851.07  5181.6 1855.86  5201.8 1863.35  5237.2 1880.46
  5242.3 1886.53  5272.6 1907.64  5363.7 1946.64  5369.7 1950.88  5404.1 1962.98
#Mann=4,-1,0
  4668.2    0.07       0  4780.8     0.1       0  5005.6    0.05       0
  5013.7     0.1       0
Bank Sta=5005.6,5013.7
Exp/Cntr=0.3,0.1

Type RM Length L Ch R = 1,35226,503,503,503
BEGIN DESCRIPTION:
Palmer Creek 69.0
END DESCRIPTION:
XS GIS Cut Line= 3
      1904224.98     13869675.02      1904575.00     13869275.00
      1904774.96     13869275.00
#Sta/Elev= 30
  4468.4 1929.25  4496.4 1925.78  4532.5 1915.40  4567.6 1887.25  4574.7 1882.75
  4581.9 1880.04  4588.5 1875.44  4602.7 1867.69  4617.0 1860.72  4631.2 1854.55
  4645.4 1850.15  4659.7 1847.56  4675.4 1846.88  4694.8 1847.68  4730.9 1846.64
  4815.3 1847.32  4886.5 1841.99  4900.8 1839.11  4992.3 1837.16  4992.8 1836.66
  5000.9 1837.16  5019.9 1838.85  5089.9 1837.51  5099.9 1839.74  5109.9 1851.98
  5119.9 1855.59  5159.9 1886.92  5169.9 1907.01  5179.9 1914.34  5199.9 1917.41
#Mann=4,-1,0
  4468.4    0.07       0  4675.4     0.1       0  4992.3    0.05       0
  5000.9     0.1       0
Bank Sta=4992.3,5000.9
Exp/Cntr=0.3,0.1

Type RM Length L Ch R = 1,34723,389,389,389
BEGIN DESCRIPTION:
Palmer Creek 68.0
END DESCRIPTION:
XS GIS Cut Line= 3
      1904474.98     13869875.03      1904650.23     13869650.20
      1904774.99     13869425.01
#Sta/Elev= 30
  4715.9 1927.35  4744.0 1924.32  4758.5 1919.79  4766.6 1918.01  4779.3 1904.77
  4787.4 1898.39  4793.7 1888.34  4808.2 1875.35  4830.0 1862.65  4851.6 1851.29
  4872.4 1845.00  4891.1 1843.79  4907.7 1844.37  4944.2 1843.56  4965.6 1839.08
  4967.6 1837.47  4968.1 1836.97  4976.3 1837.47  5000.8 1838.11  5029.8 1837.51
  5190.9 1838.30  5201.2 1840.18  5206.9 1851.39  5212.7 1875.05  5222.9 1874.70
  5228.6 1892.35  5244.7 1897.53  5250.4 1897.82  5255.6 1899.72  5258.4 1899.72
#Mann=4,-1,0
  4715.9    0.07       0  4891.1     0.1       0  4967.6    0.05       0
  4976.3     0.1       0
Bank Sta=4967.6,4976.3
Exp/Cntr=0.3,0.1

Type RM Length L Ch R = 1,34334,466,466,466
BEGIN DESCRIPTION:
Palmer Creek 67.0
END DESCRIPTION:
XS GIS Cut Line= 3
      1904874.99     13870025.04      1904925.00     13869875.00
      1905324.97     13869475.03
#Sta/Elev= 30
  4837.0 1901.21  4847.6 1901.19  4879.2 1898.26  4889.8 1895.59  4900.3 1847.73
  4922.6 1837.98  4980.3 1837.36  4980.8 1836.86  4989.0 1837.36  5051.7 1837.45
  5065.9 1839.84  5080.0 1845.38  5094.2 1841.28  5108.3 1839.22  5158.2 1839.61
  5207.3 1840.95  5235.6 1844.38  5263.9 1853.87  5304.3 1873.07  5348.7 1898.05
  5377.0 1909.40  5391.1 1916.38  5439.2 1932.42  5461.9 1938.79  5505.5 1954.25
  5518.4 1958.17  5525.5 1959.23  5532.6 1962.57  5546.7 1966.61  5560.8 1968.53
#Mann=8,-1,0
  4837.0   0.035       0  4922.6     0.1       0  4980.3    0.05       0
  4989.0     0.1       0  5158.2    0.07       0  5304.3     0.1       0
  5439.2    0.07       0  5505.5     0.1       0
Bank Sta=4980.3,4989
Exp/Cntr=0.3,0.1

Type RM Length L Ch R = 1,33868,392,392,392
BEGIN DESCRIPTION:
Palmer Creek 66.0
END DESCRIPTION:
XS GIS Cut Line= 3
      1905075.00     13870075.00      1905298.56     13870006.63
      1905475.01     13869574.98
#Sta/Elev= 30
  4685.1 1881.22  4747.8 1878.26  4772.3 1868.87  4779.2 1864.61  4831.5 1852.49
  4837.8 1844.18  4843.1 1825.11  4888.8 1821.91  4889.9 1821.81  4890.4 1821.31
  4898.6 1821.81  4953.8 1822.04  4985.5 1824.59  4996.3 1821.96  5007.2 1822.21
  5017.9 1827.14  5084.7 1832.47  5108.7 1837.28  5125.9 1846.21  5156.7 1857.93
  5210.2 1885.87  5223.1 1894.47  5233.9 1898.02  5263.6 1918.52  5293.0 1932.81
  5298.7 1937.15  5309.6 1941.11  5341.0 1960.10  5363.6 1968.44  5385.2 1970.70
#Mann=4,-1,0
  4685.1    0.07       0  4888.8     0.1       0  4889.9    0.05       0
  4898.6     0.1       0
Bank Sta=4889.9,4898.6
Exp/Cntr=0.3,0.1

Type RM Length L Ch R = 1,33476,452,452,452
BEGIN DESCRIPTION:
Palmer Creek 65.0
END DESCRIPTION:
XS GIS Cut Line= 3
      1905175.02     13870624.98      1905575.00     13870225.00
      1905774.98     13870175.00
#Sta/Elev= 30
  4433.9 1884.16  4437.4 1884.16  4448.0 1880.47  4462.2 1877.36  4490.4 1869.48
  4575.3 1848.15  4589.4 1846.16  4603.6 1844.72  4631.9 1843.41  4674.3 1836.94
  4702.6 1833.52  4745.0 1831.52  4831.8 1829.32  4914.7 1829.38  4943.0 1827.53
  4951.0 1826.33  4971.3 1823.21  4990.6 1821.93  4991.1 1821.43  5001.4 1821.93
  5112.9 1823.02  5123.3 1826.26  5133.6 1871.91  5141.3 1890.62  5146.4 1890.90
  5154.2 1902.91  5164.5 1914.85  5174.8 1918.55  5182.5 1922.44  5205.7 1923.56
#Mann=5,-1,0
  4433.9     0.1       0  4831.8    0.07       0  4951.0     0.1       0
  4990.6    0.05       0  5001.4     0.1       0
Bank Sta=4990.6,5001.4
Exp/Cntr=0.3,0.1

Type RM Length L Ch R = 1,33024,394,394,394
BEGIN DESCRIPTION:
Palmer Creek 64.0
END DESCRIPTION:
XS GIS Cut Line= 4
      1905174.97     13870675.01      1905459.87     13870603.78
      1905618.99     13870597.00      1905675.04     13870625.02
#Sta/Elev= 30
  4616.9 1885.80  4619.5 1885.80  4635.0 1879.88  4640.1 1879.43  4658.2 1870.30
  4676.2 1862.74  4681.4 1863.12  4717.4 1849.33  4722.6 1849.83  4758.7 1836.28
  4763.8 1837.18  4771.5 1834.31  4799.9 1829.49  4841.1 1827.82  4910.6 1828.17
  4925.7 1825.85  4940.3 1821.65  4940.8 1821.15  4951.1 1821.65  4997.5 1822.65
  5069.8 1823.59  5073.8 1831.57  5079.3 1833.07  5087.7 1839.97  5096.1 1875.41
  5098.9 1882.54  5101.7 1889.67  5110.1 1900.35  5118.5 1901.98  5132.5 1902.46
#Mann=5,-1,0
  4616.9     0.1       0  4940.3   0.033       0  4951.1     0.1       0
  4997.5   0.033       0  5098.9     0.1       0
Bank Sta=4940.3,4951.1
Exp/Cntr=0.3,0.1

Type RM Length L Ch R = 1,32630,439,439,439
BEGIN DESCRIPTION:
Palmer Creek 63.0
END DESCRIPTION:
XS GIS Cut Line= 3
      1905124.99     13871025.00      1905525.00     13870925.00
      1905624.98     13870875.01
#Sta/Elev= 30
  4586.8 1914.60  4603.9 1909.66  4610.0 1908.78  4617.7 1899.86  4628.0 1893.51
  4646.1 1877.73  4651.2 1877.84  4659.0 1864.11  4687.3 1847.02  4692.5 1847.36
  4710.5 1837.08  4728.5 1830.37  4782.7 1824.96  4816.2 1824.61  4852.2 1822.18
  4908.5 1822.62  4991.1 1821.38  4991.6 1820.88  5001.9 1821.38  5007.5 1823.67
  5012.0 1823.34  5029.9 1833.53  5035.5 1833.65  5052.2 1844.98  5057.8 1846.43
  5066.2 1853.04  5080.2 1856.37  5102.5 1863.79  5108.1 1867.63  5110.9 1867.63
#Mann=6,-1,0
  4586.8    0.07       0  4603.9     0.1       0  4908.5   0.033       0
  4991.1   0.033       0  5001.9   0.033       0  5012.0     0.1       0
Bank Sta=4991.1,5001.9
Exp/Cntr=0.3,0.1

Type RM Length L Ch R = 1,32191,471,471,471
BEGIN DESCRIPTION:
Palmer Creek 62.0
END DESCRIPTION:
XS GIS Cut Line= 3
      1905475.00     13871475.01      1905575.00     13871275.00
      1905774.99     13870925.02
#Sta/Elev= 30
  4771.9 1932.89  4794.3 1928.40  4816.6 1915.73  4825.0 1906.46  4839.0 1886.09
  4847.4 1865.25  4861.4 1850.79  4869.7 1827.10  4914.5 1820.15  4914.6 1818.49
  4915.1 1817.99  4925.5 1818.49  4936.8 1821.86  4942.4 1818.77  4959.2 1822.58
  4964.8 1820.39  4981.5 1822.42  5030.2 1821.98  5062.5 1824.01  5068.2 1826.27
  5099.4 1825.67  5148.8 1825.34  5192.0 1828.17  5207.9 1830.73  5256.0 1846.09
  5272.7 1853.25  5288.5 1854.65  5325.9 1870.26  5347.5 1876.20  5398.6 1881.98
#Mann=6,-1,0
  4771.9     0.1       0  4914.6    0.05       0  4925.5     0.1       0
  5030.2   0.033       0  5099.4     0.1       0  5256.0    0.07       0
Bank Sta=4914.6,4925.5
Exp/Cntr=0.3,0.1

Type RM Length L Ch R = 1,31720,419,419,419
BEGIN DESCRIPTION:
Palmer Creek 61.0
END DESCRIPTION:
XS GIS Cut Line= 3
      1905875.00     13871624.99      1905975.00     13871325.00
      1905825.01     13870925.01
#Sta/Elev= 30
  4684.1 1926.12  4726.3 1913.33  4768.4 1895.14  4779.0 1892.28  4789.5 1887.43
  4831.7 1856.15  4852.7 1836.56  4884.4 1819.85  4916.0 1810.81  4973.7 1802.95
  4974.2 1802.45  4984.7 1802.95  5076.0 1806.16  5100.9 1810.59  5107.1 1814.01
  5125.8 1820.32  5158.0 1820.57  5203.2 1820.76  5246.8 1823.93  5288.7 1835.12
  5296.7 1840.36  5302.0 1841.55  5310.0 1845.84  5320.7 1849.29  5326.9 1853.23
  5357.2 1864.80  5363.4 1869.76  5374.1 1873.81  5395.5 1878.91  5427.5 1882.12
#Mann=4,-1,0
  4684.1     0.1       0  4973.7    0.05       0  4984.7     0.1       0
  5158.0    0.07       0
Bank Sta=4973.7,4984.7
Exp/Cntr=0.3,0.1

Type RM Length L Ch R = 1,31301,428,428,428
BEGIN DESCRIPTION:
Palmer Creek 60.0
END DESCRIPTION:
XS GIS Cut Line= 3
      1906475.01     13871425.02      1906278.91     13871142.65
      1906225.00     13870774.97
#Sta/Elev= 30
  4712.3 1911.12  4740.7 1910.01  4748.9 1904.63  4770.4 1894.53  4791.3 1887.32
  4797.6 1880.20  4806.2 1848.19  4812.3 1847.54  4842.0 1825.98  4862.9 1814.92
  4870.6 1808.81  4883.9 1804.82  4914.1 1803.16  4914.6 1802.66  4925.3 1803.16
  5073.9 1804.14  5084.0 1806.70  5104.2 1815.60  5113.4 1818.28  5129.9 1819.95
  5306.4 1821.06  5329.7 1826.50  5346.8 1833.00  5377.1 1847.61  5387.2 1853.52
  5392.8 1858.34  5397.8 1859.32  5407.5 1864.25  5425.1 1876.77  5427.7 1876.77
#Mann=5,-1,0
  4712.3     0.1       0  4914.1    0.05       0  4925.3     0.1       0
  5129.9   0.035       0  5329.7     0.1       0
Bank Sta=4914.1,4925.3
Exp/Cntr=0.3,0.1

Type RM Length L Ch R = 1,30873,462,462,462
BEGIN DESCRIPTION:
Palmer Creek 59.0
END DESCRIPTION:
XS GIS Cut Line= 3
      1906625.00     13871275.00      1906625.00     13871125.00
      1906275.01     13870725.01
#Sta/Elev= 30
  4855.1 1892.77  4885.1 1885.13  4895.1 1880.85  4905.1 1868.87  4915.1 1860.91
  4925.1 1849.51  4935.1 1836.00  4955.1 1820.96  4965.1 1810.88  4979.5 1803.21
  4980.0 1802.71  4990.7 1803.21  5065.2 1803.69  5125.2 1803.95  5139.4 1808.26
  5147.0 1812.28  5165.7 1815.11  5281.8 1815.79  5345.4 1822.81  5380.5 1824.67
  5394.7 1827.16  5409.0 1833.36  5454.4 1858.15  5472.5 1866.90  5480.1 1873.58
  5486.8 1875.88  5494.4 1883.88  5501.0 1885.89  5508.6 1890.93  5536.6 1898.26
#Mann=6,-1,0
  4855.1     0.1       0  4979.5    0.05       0  4990.7     0.1       0
  5065.2   0.033       0  5165.7   0.035       0  5454.4     0.1       0
Bank Sta=4979.5,4990.7
Exp/Cntr=0.3,0.1

Type RM Length L Ch R = 1,30411,420,420,420
BEGIN DESCRIPTION:
Palmer Creek 58.0
END DESCRIPTION:
XS GIS Cut Line= 3
      1907025.00     13871225.03      1906975.00     13870875.00
      1906875.00     13870475.00
#Sta/Elev= 30
  4646.6 1880.28  4687.0 1874.03  4778.0 1845.69  4818.4 1835.75  4879.0 1813.61
  4899.2 1810.46  4949.7 1808.15  4959.8 1804.97  4969.9 1794.23  5012.6 1790.48
  5013.1 1789.98  5023.9 1790.48  5041.4 1794.15  5059.5 1795.26  5072.3 1798.61
  5104.5 1801.19  5184.4 1817.53  5188.3 1818.22  5229.5 1839.70  5257.9 1857.46
  5265.6 1864.00  5270.8 1865.29  5299.1 1884.87  5306.8 1891.67  5312.0 1893.08
  5340.3 1911.01  5389.3 1936.62  5394.5 1937.92  5409.9 1947.52  5412.5 1947.52
#Mann=5,-1,0
  4646.6     0.1       0  5012.6    0.05       0  5023.9     0.1       0
  5104.5   0.035       0  5184.4     0.1       0
Bank Sta=5012.6,5023.9
Exp/Cntr=0.3,0.1

Type RM Length L Ch R = 1,29991,451,451,451
BEGIN DESCRIPTION:
Palmer Creek 57.0
END DESCRIPTION:
XS GIS Cut Line= 3
      1907136.54     13871246.57      1907325.00     13870775.00
      1907474.98     13870575.03
#Sta/Elev= 30
  4491.6 1880.72  4514.8 1876.64  4529.4 1872.43  4553.7 1862.18  4607.5 1844.43
  4666.8 1829.33  4739.5 1815.04  4751.7 1811.45  4769.1 1808.93  4828.4 1806.13
  4924.1 1807.14  4977.9 1798.10  4984.6 1792.05  4991.1 1789.64  4991.6 1789.14
  5002.4 1789.64  5056.7 1790.51  5077.6 1798.03  5092.1 1805.08  5106.7 1816.79
  5113.0 1820.11  5127.6 1832.82  5135.9 1869.32  5142.1 1886.46  5149.4 1910.72
  5156.7 1916.08  5163.0 1922.51  5206.7 1950.75  5221.3 1962.93  5249.4 1963.94
#Mann=3,-1,0
  4491.6     0.1       0  4991.1    0.05       0  5002.4     0.1       0
Bank Sta=4991.1,5002.4
Exp/Cntr=0.3,0.1

Type RM Length L Ch R = 1,29540,444,444,444
BEGIN DESCRIPTION:
Palmer Creek 56.0
END DESCRIPTION:
XS GIS Cut Line= 3
      1907225.01     13871324.99      1907475.00     13871125.00
      1907675.01     13870924.99
#Sta/Elev= 30
  4675.1 1882.55  4696.7 1880.78  4711.1 1877.64  4717.5 1874.65  4725.5 1872.52
  4767.1 1852.35  4795.9 1841.19  4824.8 1828.53  4867.2 1814.50  4888.8 1809.73
  4903.2 1808.12  4931.2 1807.27  4938.4 1805.93  4944.8 1798.52  4952.8 1791.97
  5003.7 1789.90  5004.2 1789.40  5015.1 1789.90  5037.7 1790.93  5051.8 1790.40
  5094.2 1790.89  5122.5 1796.56  5136.7 1800.67  5150.8 1810.01  5179.1 1827.14
  5207.4 1847.44  5221.5 1895.74  5235.7 1905.17  5274.5 1917.39  5278.1 1917.39
#Mann=3,-1,0
  4675.1     0.1       0  5003.7    0.05       0  5015.1     0.1       0
Bank Sta=5003.7,5015.1
Exp/Cntr=0.3,0.1

Type RM Length L Ch R = 1,29096,453,453,453
BEGIN DESCRIPTION:
Palmer Creek 55.0
END DESCRIPTION:
XS GIS Cut Line= 3
      1907374.98     13871575.01      1907775.00     13871425.00
      1908075.04     13871374.99
#Sta/Elev= 30
  4577.1 1885.44  4592.3 1883.83  4617.2 1876.12  4641.2 1863.71  4647.4 1858.38
  4677.7 1844.14  4683.9 1839.66  4716.0 1823.37  4732.9 1815.62  4757.8 1807.22
  4780.0 1803.62  4823.7 1801.36  4843.2 1800.66  4865.5 1801.99  4873.5 1799.74
  4878.8 1793.26  4886.8 1791.43  4977.3 1790.10  4977.8 1789.60  4988.7 1790.10
  5075.3 1798.65  5126.0 1812.13  5146.3 1819.78  5153.9 1824.00  5158.9 1824.15
  5214.7 1852.56  5219.8 1853.75  5247.6 1869.81  5288.2 1888.91  5308.5 1893.66
#Mann=3,-1,0
  4577.1     0.1       0  4977.3    0.05       0  4988.7     0.1       0
Bank Sta=4977.3,4988.7
Exp/Cntr=0.3,0.1

Type RM Length L Ch R = 1,28643,439,439,439
BEGIN DESCRIPTION:
Palmer Creek 54.0
END DESCRIPTION:
XS GIS Cut Line= 3
      1907774.97     13872075.04      1907975.00     13871775.00
      1908225.03     13871524.97
#Sta/Elev= 30
  4639.2 1893.65  4642.3 1893.65  4646.8 1891.51  4667.8 1889.16  4697.8 1882.57
  4718.9 1869.60  4739.9 1858.83  4754.9 1848.14  4769.9 1841.44  4791.0 1829.61
  4827.0 1813.09  4842.1 1808.43  4863.1 1803.59  4914.2 1798.22  4941.2 1794.36
  4956.2 1790.90  4990.8 1790.24  4991.3 1789.74  5002.7 1790.24  5084.7 1790.33
  5098.8 1795.57  5155.4 1798.32  5183.7 1805.96  5211.9 1817.64  5240.2 1831.91
  5268.5 1849.79  5310.9 1879.10  5325.1 1885.81  5339.2 1890.30  5353.4 1891.65
#Mann=3,-1,0
  4639.2     0.1       0  4990.8    0.05       0  5002.7     0.1       0
Bank Sta=4990.8,5002.7
Exp/Cntr=0.3,0.1

Type RM Length L Ch R = 1,28204,459,459,459
BEGIN DESCRIPTION:
Palmer Creek 53.0
END DESCRIPTION:
XS GIS Cut Line= 3
      1908025.00     13872275.00      1908275.00     13871975.00
      1908374.99     13871625.02
#Sta/Elev= 30
  4608.7 1899.88  4644.5 1892.83  4673.1 1885.14  4686.8 1876.33  4694.0 1867.81
  4700.5 1863.02  4751.2 1830.74  4786.4 1812.58  4800.7 1807.45  4821.5 1802.81
  4843.0 1800.82  4864.5 1791.90  4878.8 1790.50  5010.2 1789.72  5010.7 1789.22
  5022.1 1789.72  5030.4 1793.49  5055.1 1794.55  5155.2 1796.28  5176.0 1800.33
  5200.7 1807.88  5207.2 1811.95  5228.0 1820.26  5259.2 1835.11  5300.8 1857.85
  5307.3 1863.98  5321.6 1870.93  5332.0 1877.80  5341.1 1880.71  5363.2 1882.56
#Mann=4,-1,0
  4608.7     0.1       0  5010.2    0.05       0  5022.1     0.1       0
  5055.1     0.1       0
Bank Sta=5010.2,5022.1
Exp/Cntr=0.3,0.1

Type RM Length L Ch R = 1,27745,412,412,412
BEGIN DESCRIPTION:
Palmer Creek 52.0
END DESCRIPTION:
XS GIS Cut Line= 3
      1908625.00     13872425.00      1908625.00     13872125.00
      1908425.00     13871725.01
#Sta/Elev= 30
  4707.8 1907.15  4717.8 1905.21  4747.8 1884.98  4757.8 1870.83  4767.8 1859.66
  4777.8 1841.87  4787.8 1833.11  4817.8 1815.27  4827.8 1810.76  4837.8 1809.24
  4887.8 1807.50  4917.8 1797.62  4927.8 1790.60  4931.8 1785.19  4932.3 1784.69
  4943.8 1785.19  4991.2 1785.58  5111.2 1785.44  5128.0 1789.06  5133.6 1786.97
  5142.0 1792.15  5150.3 1793.89  5298.5 1796.00  5339.0 1802.10  5379.5 1813.02
  5396.3 1821.20  5424.3 1829.56  5441.0 1839.77  5446.6 1840.16  5455.0 1844.55
#Mann=5,-1,0
  4707.8     0.1       0  4931.8    0.05       0  4943.8     0.1       0
  4991.2    0.07       0  5339.0     0.1       0
Bank Sta=4931.8,4943.8
Exp/Cntr=0.3,0.1

Type RM Length L Ch R = 1,27333,471,471,471
BEGIN DESCRIPTION:
Palmer Creek 51.0
END DESCRIPTION:
XS GIS Cut Line= 3
      1909025.00     13872374.99      1908975.00     13872125.00
      1908825.02     13871725.04
#Sta/Elev= 30
  4749.2 1887.67  4769.6 1884.64  4779.8 1850.96  4790.0 1832.58  4820.6 1814.40
  4830.8 1809.98  4861.4 1798.05  4871.6 1797.68  4902.2 1786.26  4988.9 1785.28
  4995.5 1785.15  4996.0 1784.65  5007.6 1785.15  5025.5 1785.62  5044.2 1789.72
  5094.5 1790.73  5159.9 1793.23  5270.3 1795.41  5325.3 1798.92  5345.9 1803.20
  5355.7 1806.69  5361.0 1807.15  5367.3 1812.11  5386.0 1821.44  5391.3 1822.02
  5410.0 1831.12  5416.2 1835.47  5421.6 1835.48  5428.7 1839.94  5431.3 1839.94
#Mann=6,-1,0
  4749.2     0.1       0  4988.9   0.033       0  4995.5   0.033       0
  5007.6   0.033       0  5094.5    0.07       0  5325.3     0.1       0
Bank Sta=4995.5,5007.6
Exp/Cntr=0.3,0.1

Type RM Length L Ch R = 1,26862,482,482,482
BEGIN DESCRIPTION:
Palmer Creek 50.0
END DESCRIPTION:
XS GIS Cut Line= 3
      1909280.38     13872425.15      1909375.00     13872025.00
      1909317.41     13871529.11
#Sta/Elev= 30
  4594.3 1861.90  4615.0 1860.41  4645.8 1852.08  4697.2 1844.20  4707.5 1834.73
  4723.0 1814.93  4728.1 1816.15  4736.3 1810.98  4748.6 1803.63  4812.7 1803.73
  4820.5 1800.16  4841.1 1796.87  4849.8 1792.66  4854.9 1793.61  4871.9 1786.14
  4968.6 1784.49  4969.1 1783.99  4980.7 1784.49  5075.4 1788.84  5216.9 1789.38
  5271.3 1794.05  5337.7 1811.75  5367.9 1822.18  5408.2 1842.27  5418.2 1849.07
  5428.3 1856.99  5438.4 1870.45  5468.6 1892.56  5488.7 1899.95  5504.7 1902.13
#Mann=6,-1,0
  4594.3     0.1       0  4736.3    0.07       0  4968.6   0.033       0
  4980.7    0.07       0  5075.4    0.07       0  5271.3     0.1       0
Bank Sta=4968.6,4980.7
Exp/Cntr=0.3,0.1

Type RM Length L Ch R = 1,26380,406,406,406
BEGIN DESCRIPTION:
Palmer Creek 49.0
END DESCRIPTION:
XS GIS Cut Line= 3
      1909474.98     13872225.01      1909825.00     13871925.00
      1909925.01     13871774.98
#Sta/Elev= 30
  4543.2 1807.94  4564.6 1806.76  4624.8 1797.43  4636.6 1796.05  4663.4 1793.84
  4691.9 1788.78  4706.2 1785.29  4720.5 1785.89  4776.3 1785.43  4806.1 1784.49
  4962.4 1784.23  4962.9 1783.73  4974.6 1784.23  4990.5 1785.01  5000.9 1788.30
  5007.2 1788.30  5017.7 1793.80  5026.7 1795.82  5040.3 1801.66  5047.8 1806.57
  5053.8 1809.17  5068.8 1817.48  5076.3 1823.36  5098.8 1838.81  5104.9 1843.42
  5112.4 1851.18  5134.9 1868.03  5155.9 1887.80  5171.0 1894.52  5184.5 1895.62
#Mann=6,-1,0
  4543.2   0.035       0  4624.8    0.07       0  4636.6   0.035       0
  4776.3   0.033       0  4962.4   0.033       0  4974.6   0.033       0
Bank Sta=4962.4,4974.6
Exp/Cntr=0.3,0.1

Type RM Length L Ch R = 1,25974,329,329,329
BEGIN DESCRIPTION:
Palmer Creek 48.0
END DESCRIPTION:
XS GIS Cut Line= 3
      1909575.01     13872574.99      1909983.23     13872272.64
      1910275.03     13872174.99
#Sta/Elev= 30
  4504.9 1829.56  4508.0 1829.56  4512.2 1827.10  4550.0 1821.63  4576.9 1815.20
  4597.8 1806.60  4618.6 1803.41  4647.8 1802.45  4654.2 1803.74  4662.5 1802.56
  4668.7 1803.32  4697.9 1798.87  4741.3 1797.84  4748.0 1795.52  4768.9 1794.03
  4783.5 1790.77  4819.0 1787.46  4883.7 1785.17  5008.3 1784.43  5061.4 1784.32
  5061.9 1783.82  5073.6 1784.32  5241.6 1784.96  5257.3 1788.42  5267.8 1795.19
  5273.2 1801.78  5278.5 1803.44  5288.9 1842.55  5299.5 1877.07  5320.6 1875.23
#Mann=5,-1,0
  4504.9    0.07       0  4550.0   0.035       0  5008.3   0.033       0
  5061.4   0.035       0  5073.6   0.033       0
Bank Sta=5061.4,5073.6
Exp/Cntr=0.3,0.1

Type RM Length L Ch R = 1,25645,213,213,213
BEGIN DESCRIPTION:
Palmer Creek 47.0
END DESCRIPTION:
XS GIS Cut Line= 3
      1909506.72     13872628.16      1909993.48     13872521.36
      1910325.02     13872274.99
#Sta/Elev= 30
  4374.7 1848.23  4403.7 1842.36  4410.8 1839.09  4415.9 1839.98  4454.6 1825.74
  4459.7 1826.26  4485.6 1817.10  4516.3 1816.43  4559.0 1809.64  4618.7 1803.63
  4645.2 1803.60  4689.0 1797.63  4737.9 1786.87  4823.8 1786.43  4907.5 1786.81
  4942.9 1784.30  5001.5 1784.18  5002.0 1783.68  5013.7 1784.18  5030.7 1784.33
  5117.8 1784.46  5199.5 1785.35  5214.1 1790.99  5222.5 1797.75  5228.7 1800.09
  5236.2 1823.81  5243.3 1850.43  5249.5 1854.24  5264.4 1856.77  5286.1 1855.46
#Mann=8,-1,0
  4374.7    0.07       0  4559.0   0.035       0  4823.8    0.07       0
  5001.5    0.05       0  5013.7    0.07       0  5030.7   0.035       0
  5117.8   0.033       0  5264.4     0.1       0
Bank Sta=5001.5,5013.7
Exp/Cntr=0.3,0.1

Type RM Length L Ch R = 1,25432,122,122,122
BEGIN DESCRIPTION:
Palmer Creek D1
END DESCRIPTION:
XS GIS Cut Line= 5
      1909586.53     13872862.23      1909905.96     13872580.99
      1910149.01     13872521.97      1910291.37     13872504.61
      1910360.41     13872363.07
#Sta/Elev= 30
  4213.6 1882.91  4217.6 1880.49  4246.1 1875.58  4281.2 1861.30  4395.0 1824.22
  4437.7 1817.08  4472.8 1816.26  4487.0 1810.95  4521.3 1805.88  4550.6 1800.77
  4571.5 1801.39  4621.7 1785.77  4704.0 1786.50  4782.3 1785.90  4852.2 1794.12
  4979.8 1793.11  5043.4 1792.84  5050.7 1789.72  5063.0 1789.06  5081.8 1785.39
  5082.3 1784.89  5094.0 1785.39  5110.2 1791.82  5123.8 1800.22  5132.4 1814.06
  5140.8 1821.62  5163.3 1827.70  5170.8 1827.02  5185.9 1831.29  5190.2 1829.38
#Mann=8,-1,0
  4213.6    0.07       0  4521.3   0.035       0  4704.0    0.07       0
  4979.8   0.035       0  5063.0     0.1       0  5081.8   0.035       0
  5094.0     0.1       0  5170.8     0.1       0
Bank Sta=5081.8,5094
Exp/Cntr=0.3,0.1

Type RM Length L Ch R = 1,25310,316,316,316
BEGIN DESCRIPTION:
Palmer Creek 46.1
END DESCRIPTION:
XS GIS Cut Line= 4
      1909653.63     13872894.12      1910250.38     13872629.24
      1910612.12     13872573.82      1910995.87     13872271.47
#Sta/Elev= 30
  4317.6 1881.87  4349.4 1876.26  4354.9 1872.77  4372.7 1872.60  4378.2 1866.76
  4401.4 1865.32  4494.2 1836.06  4523.2 1822.52  4559.8 1812.54  4650.5 1793.86
  4680.1 1784.27  4696.1 1782.79  4772.6 1779.62  4833.3 1778.87  4870.8 1783.38
  4922.8 1776.81  4969.4 1767.10  5025.1 1765.52  5025.6 1765.02  5037.3 1765.52
  5066.2 1773.52  5097.2 1776.01  5137.0 1779.18  5218.0 1773.87  5278.7 1780.78
  5588.7 1798.07  5671.6 1805.70  5735.8 1817.58  5780.5 1829.42  5825.0 1842.47
#Mann=8,-1,0
  4317.6    0.07       0  4696.1   0.035       0  4772.6    0.07       0
  5025.1    0.05       0  5037.3    0.07       0  5097.2    0.07       0
  5588.7   0.035       0  5780.5     0.1       0
Bank Sta=5025.1,5037.3
Exp/Cntr=0.3,0.1

Type RM Length L Ch R = 1,24994,471,471,471
BEGIN DESCRIPTION:
Palmer Creek 46.0
END DESCRIPTION:
XS GIS Cut Line= 3
      1910034.61     13873143.06      1910325.00     13872925.00
      1911079.26     13872230.29
#Sta/Elev= 30
  4637.4 1888.18  4672.5 1883.88  4700.6 1862.69  4707.9 1858.49  4722.5 1842.31
  4728.7 1831.04  4737.1 1829.17  4743.3 1820.44  4757.9 1816.71  4764.1 1810.71
  4778.7 1806.01  4828.7 1803.68  4857.9 1793.23  4922.4 1779.71  4949.0 1769.42
  4986.8 1760.39  4987.3 1759.89  4999.8 1760.39  5057.0 1761.18  5078.5 1771.40
  5092.7 1772.98  5340.4 1777.63  5573.6 1792.98  5657.5 1795.31  5757.9 1801.07
  5828.8 1814.19  5882.7 1829.07  5984.2 1858.05  5991.6 1863.60  6026.0 1867.61
#Mann=7,-1,0
  4637.4    0.07       0  4700.6     0.1       0  4949.0    0.07       0
  4986.8    0.05       0  4999.8    0.07       0  5657.5   0.035       0
  5882.7     0.1       0
Bank Sta=4986.8,4999.8
Exp/Cntr=0.3,0.1

Type RM Length L Ch R = 1,24523,472,472,472
BEGIN DESCRIPTION:
Palmer Creek 45.0
END DESCRIPTION:
XS GIS Cut Line= 3
      1910619.40     13873731.06      1910625.00     13873275.00
      1911241.05     13872445.66
#Sta/Elev= 30
  4539.8 1843.50  4555.9 1832.65  4575.9 1825.13  4675.9 1822.74  4799.5 1804.02
  4865.9 1800.58  4885.9 1798.29  4897.9 1793.97  4905.9 1792.78  4915.9 1786.45
  4925.9 1776.21  4945.9 1774.09  4975.9 1757.26  4996.5 1756.26  4997.0 1755.76
  5009.9 1756.26  5038.7 1757.02  5055.1 1760.77  5124.2 1776.72  5296.7 1778.34
  5341.7 1777.35  5460.0 1775.12  5831.4 1777.15  5860.6 1779.38  5875.2 1787.86
  5930.5 1807.39  5960.7 1816.97  5975.4 1825.11  6010.8 1838.98  6029.0 1850.29
#Mann=9,-1,0
  4539.8    0.07       0  4799.5   0.035       0  4897.9    0.07       0
  4996.5    0.05       0  5009.9    0.07       0  5055.1    0.07       0
  5296.7   0.035       0  5341.7    0.07       0  5930.5     0.1       0
Bank Sta=4996.5,5009.9
Exp/Cntr=0.3,0.1

Type RM Length L Ch R = 1,24051,407,407,407
BEGIN DESCRIPTION:
Palmer Creek 44.0
END DESCRIPTION:
XS GIS Cut Line= 3
      1911075.00     13873625.01      1911025.00     13873375.00
      1911280.49     13872456.75
#Sta/Elev= 30
  4753.0 1851.88  4783.6 1846.56  4793.8 1843.06  4804.0 1827.15  4834.6 1803.20
  4844.8 1794.16  4855.0 1782.26  4878.8 1763.37  4895.8 1757.77  4970.6 1756.39
  4971.1 1755.89  4984.1 1756.39  5005.4 1764.29  5010.6 1764.29  5018.3 1768.73
  5080.6 1774.55  5138.1 1776.36  5163.7 1775.33  5477.3 1773.46  5786.5 1775.17
  5796.8 1775.73  5806.0 1778.09  5828.0 1786.01  5846.1 1795.29  5850.6 1795.95
  5879.7 1810.03  5884.9 1810.82  5890.3 1815.31  5952.5 1846.18  5961.1 1852.93
#Mann=5,-1,0
  4753.0   0.035       0  4878.8    0.07       0  4970.6    0.05       0
  4984.1    0.07       0  5846.1     0.1       0
Bank Sta=4970.6,4984.1
Exp/Cntr=0.3,0.1

Type RM Length L Ch R = 1,23644,542,542,542
BEGIN DESCRIPTION:
Palmer Creek 43.0
END DESCRIPTION:
XS GIS Cut Line= 3
      1911425.00     13873575.00      1911384.74     13873261.21
      1911675.00     13872724.99
#Sta/Elev= 30
  4777.1 1845.83  4807.3 1841.39  4814.4 1837.42  4819.4 1837.55  4827.5 1829.22
  4837.6 1816.03  4877.9 1783.51  4885.2 1774.31  4894.0 1762.33  4908.2 1757.70
  4990.7 1756.45  4992.2 1756.38  4992.7 1755.88  5005.7 1756.38  5019.1 1759.50
  5059.4 1765.02  5105.4 1766.59  5121.5 1768.87  5127.2 1768.27  5143.4 1771.28
  5180.1 1772.43  5230.9 1770.65  5378.4 1769.51  5569.5 1769.60  5645.7 1773.32
  5655.6 1776.80  5673.2 1782.98  5695.1 1794.27  5700.3 1798.44  5703.2 1798.44
#Mann=6,-1,0
  4777.1    0.07       0  4885.2     0.1       0  4990.7    0.07       0
  4992.2    0.05       0  5005.7    0.07       0  5655.6     0.1       0
Bank Sta=4992.2,5005.7
Exp/Cntr=0.3,0.1

Type RM Length L Ch R = 1,23102,447,447,447
BEGIN DESCRIPTION:
Palmer Creek 42.0
END DESCRIPTION:
XS GIS Cut Line= 3
      1911837.45     13873518.64      1911808.46     13873114.77
      1911869.83     13872698.89
#Sta/Elev= 30
  4654.9 1783.71  4756.4 1773.19  4761.4 1775.25  4795.6 1769.80  4909.2 1751.11
  4929.2 1749.21  4969.3 1748.85  4989.4 1747.29  5002.7 1743.98  5003.2 1743.48
  5016.2 1743.98  5019.5 1744.10  5029.5 1755.27  5062.2 1761.52  5067.5 1764.06
  5072.5 1763.20  5087.2 1766.21  5241.5 1765.92  5271.3 1768.33  5302.2 1775.48
  5322.4 1783.69  5341.0 1796.04  5346.0 1797.77  5352.7 1803.47  5403.3 1832.97
  5410.6 1840.21  5453.8 1868.16  5463.9 1877.69  5474.0 1884.38  5480.2 1894.14
#Mann=5,-1,0
  4654.9   0.035       0  4795.6    0.07       0  5002.7    0.05       0
  5016.2    0.07       0  5087.2     0.1       0
Bank Sta=5002.7,5016.2
Exp/Cntr=0.3,0.1

Type RM Length L Ch R = 1,22655,437,437,437
BEGIN DESCRIPTION:
Palmer Creek 41.0
END DESCRIPTION:
XS GIS Cut Line= 3
      1912075.01     13873324.99      1912225.00     13873175.00
      1912375.03     13873024.97
#Sta/Elev= 30
  4787.6 1768.78  4811.2 1768.48  4844.2 1767.78  4872.4 1766.30  4914.9 1761.73
  4929.0 1761.24  4943.2 1759.63  4957.3 1750.23  4971.4 1744.74  4985.6 1747.18
  5003.3 1747.80  5013.9 1746.59  5021.2 1742.27  5021.7 1741.77  5034.3 1741.77
  5034.8 1742.27  5042.1 1746.24  5056.3 1752.08  5059.1 1752.75  5070.4 1755.46
  5084.6 1763.71  5112.9 1778.83  5127.0 1788.30  5141.1 1796.08  5155.3 1807.00
  5169.4 1874.58  5183.6 1884.65  5197.7 1889.58  5208.3 1891.31  5211.9 1891.31
#Mann=5,-1,0
  4787.6     0.1       0  4811.2    0.07       0  5021.2    0.05       0
  5034.8    0.07       0  5059.1     0.1       0
Bank Sta=5021.2,5034.8
Exp/Cntr=0.3,0.1

Type RM Length L Ch R = 1,22218,437,437,437
BEGIN DESCRIPTION:
Palmer Creek 40.0
END DESCRIPTION:
XS GIS Cut Line= 3
      1912174.95     13873525.00      1912375.00     13873525.00
      1912575.00     13873275.00
#Sta/Elev= 30
  4805.0 1766.78  4882.8 1765.21  4905.0 1764.26  4935.9 1758.42  4955.0 1753.96
  4995.7 1740.34  4996.2 1739.84  5009.4 1740.34  5018.7 1744.16  5076.3 1744.90
  5090.7 1747.84  5119.5 1749.24  5126.6 1751.68  5140.3 1754.72  5169.1 1771.73
  5175.5 1778.29  5183.5 1780.45  5189.9 1788.24  5197.1 1789.32  5210.7 1800.32
  5218.8 1804.17  5225.2 1811.83  5239.6 1821.01  5247.6 1824.12  5254.0 1831.34
  5268.4 1841.65  5274.8 1850.81  5297.2 1866.25  5303.6 1869.69  5325.2 1875.49
#Mann=6,-1,0
  4805.0     0.1       0  4882.8   0.035       0  4935.9    0.07       0
  4995.7    0.05       0  5009.4    0.07       0  5126.6     0.1       0
Bank Sta=4995.7,5009.4
Exp/Cntr=0.3,0.1

Type RM Length L Ch R = 1,21781,476,476,476
BEGIN DESCRIPTION:
Palmer Creek 39.0
END DESCRIPTION:
XS GIS Cut Line= 4
      1912374.97     13873975.01      1912547.07     13873931.98
      1912592.36     13873867.14      1912725.00     13873425.00
#Sta/Elev= 30
  4774.9 1769.47  4921.8 1761.48  4940.5 1753.77  4948.7 1748.97  4952.3 1748.97
  4956.1 1745.10  4959.2 1744.24  4991.1 1738.97  4991.6 1738.47  5004.8 1738.97
  5029.6 1743.17  5075.4 1745.42  5117.1 1745.73  5158.0 1748.82  5172.3 1751.78
  5202.6 1757.40  5221.5 1760.33  5267.7 1774.83  5273.7 1778.25  5284.2 1781.64
  5326.0 1790.26  5339.0 1795.71  5372.1 1803.72  5388.6 1812.60  5399.0 1816.23
  5411.4 1818.20  5443.4 1822.97  5471.2 1829.36  5476.5 1828.52  5493.0 1833.13
#Mann=8,-1,0
  4774.9   0.035       0  4940.5     0.1       0  4959.2    0.07       0
  4991.1    0.05       0  5004.8    0.07       0  5172.3     0.1       0
  5202.6    0.07       0  5411.4     0.1       0
Bank Sta=4991.1,5004.8
Exp/Cntr=0.3,0.1

Type RM Length L Ch R = 1,21305,442,442,442
BEGIN DESCRIPTION:
Palmer Creek 38.0
END DESCRIPTION:
XS GIS Cut Line= 4
      1912575.02     13874374.99      1912825.00     13874275.00
      1913025.00     13874125.00      1913225.79     13873890.04
#Sta/Elev= 30
  4731.2 1774.45  4763.5 1771.80  4794.5 1767.49  4824.1 1760.93  4902.2 1755.04
  4907.5 1755.41  4925.0 1752.47  4931.8 1749.81  4937.2 1751.52  4956.0 1744.46
  4961.4 1744.33  4968.1 1741.47  4978.9 1740.68  4997.7 1736.41  5015.3 1736.14
  5015.8 1735.64  5029.3 1736.14  5043.1 1739.71  5050.4 1739.29  5061.7 1740.54
  5072.3 1741.82  5136.9 1744.01  5150.4 1746.50  5164.0 1750.63  5172.3 1751.70
  5186.9 1752.09  5246.9 1758.03  5359.5 1760.89  5470.6 1763.87  5559.5 1764.93
#Mann=6,-1,0
  4731.2   0.035       0  5015.3   0.035       0  5029.3   0.035       0
  5061.7    0.07       0  5246.9   0.035       0  5359.5    0.07       0
Bank Sta=5015.3,5029.3
Exp/Cntr=0.3,0.1

Type RM Length L Ch R = 1,20863,414,414,414
BEGIN DESCRIPTION:
Palmer Creek 37.0
END DESCRIPTION:
XS GIS Cut Line= 4
      1913125.00     13875124.97      1913175.00     13874525.00
      1913286.33     13873914.19      1913351.94     13873511.32
#Sta/Elev= 30
  4393.2 1862.82  4450.9 1845.35  4455.9 1845.70  4520.9 1821.70  4571.3 1803.37
  4603.9 1794.02  4613.9 1786.06  4674.1 1772.72  4764.5 1769.54  4784.5 1766.58
  4804.6 1760.02  4824.7 1749.32  4862.8 1743.24  4894.9 1739.27  4978.2 1734.82
  4978.7 1734.32  4992.3 1734.82  5021.9 1735.49  5046.1 1747.16  5056.2 1749.43
  5086.7 1748.99  5182.5 1756.88  5208.8 1755.89  5437.4 1759.16  5701.3 1765.95
  5797.7 1780.15  5838.2 1783.92  5895.4 1796.49  5919.3 1801.08  6024.3 1831.77
#Mann=9,-1,0
  4393.2    0.07       0  4520.9   0.035       0  4862.8    0.07       0
  4978.2    0.05       0  4992.3    0.07       0  5182.5    0.07       0
  5208.8   0.035       0  5437.4    0.07       0  5895.4     0.1       0
Bank Sta=4978.2,4992.3
Exp/Cntr=0.3,0.1

Type RM Length L Ch R = 1,20449,432,432,432
BEGIN DESCRIPTION:
Palmer Creek 36.0
END DESCRIPTION:
XS GIS Cut Line= 4
      1913325.00     13874925.00      1913475.00     13874775.00
      1913681.68     13874161.01      1913808.81     13873618.78
#Sta/Elev= 30
  4783.7 1805.38  4812.0 1799.88  4826.1 1794.68  4840.3 1784.98  4868.5 1785.89
  4882.7 1788.35  4889.8 1787.26  4911.0 1760.24  4925.1 1745.32  4939.3 1736.91
  4974.6 1732.54  4975.1 1732.04  4988.7 1732.54  4992.3 1734.76  5006.3 1735.10
  5027.5 1732.92  5069.3 1743.69  5122.4 1745.76  5154.1 1751.34  5175.2 1753.02
  5289.8 1753.95  5387.8 1752.53  5725.4 1751.95  5900.6 1756.58  5947.9 1758.67
  6075.2 1770.00  6111.3 1776.87  6142.9 1784.51  6194.2 1802.31  6200.6 1805.84
#Mann=6,-1,0
  4783.7    0.07       0  4974.6    0.05       0  4988.7    0.07       0
  5387.8   0.035       0  5900.6    0.07       0  6111.3     0.1       0
Bank Sta=4974.6,4988.7
Exp/Cntr=0.3,0.1

Type RM Length L Ch R = 1,20017,471,471,471
BEGIN DESCRIPTION:
Palmer Creek 35.0
END DESCRIPTION:
XS GIS Cut Line= 5
      1913313.45     13875000.00      1913799.03     13874972.06
      1913825.00     13874925.00      1913869.91     13874220.45
      1913871.42     13873633.56
#Sta/Elev= 30
  4459.8 1821.81  4501.4 1817.43  4561.5 1797.63  4601.6 1793.01  4630.3 1787.10
  4651.7 1787.05  4721.8 1779.99  4771.9 1767.54  4807.4 1762.12  4922.1 1756.66
  4932.1 1753.66  4948.4 1755.82  4954.2 1754.71  4977.1 1734.79  5012.9 1732.60
  5013.4 1732.10  5027.0 1732.60  5072.0 1735.86  5137.6 1738.81  5295.5 1744.76
  5380.3 1745.10  5420.8 1746.12  5470.9 1751.34  5570.1 1751.17  5861.4 1749.87
  6044.5 1756.26  6141.4 1764.81  6191.4 1774.67  6236.4 1788.98  6292.8 1807.77
#Mann=10,-1,0
  4459.8    0.07       0  5012.9    0.05       0  5027.0    0.07       0
  5072.0     0.1       0  5137.6    0.07       0  5295.5   0.035       0
  5380.3    0.07       0  5570.1   0.035       0  6044.5    0.07       0
  6236.4     0.1       0
Bank Sta=5012.9,5027
Exp/Cntr=0.3,0.1

Type RM Length L Ch R = 1,19546,360,360,360
BEGIN DESCRIPTION:
Palmer Creek 34.0
END DESCRIPTION:
XS GIS Cut Line= 3
      1914375.02     13875125.04      1914225.00     13874825.00
      1913904.79     13873648.76
#Sta/Elev= 30
  4664.5 1760.28  4675.0 1760.01  4700.9 1757.92  4717.7 1750.93  4740.0 1745.41
  4842.6 1745.63  4863.1 1745.85  4888.2 1745.48  4896.5 1737.88  4910.5 1732.51
  4982.7 1732.37  4983.2 1731.87  5000.4 1732.37  5060.9 1737.04  5170.3 1740.57
  5272.5 1741.67  5359.0 1740.41  5416.3 1747.62  5456.0 1750.74  5575.4 1749.44
  5758.6 1748.83  5793.0 1748.83  5912.0 1750.98  5986.6 1756.31  6049.4 1761.82
  6123.7 1775.41  6163.5 1787.68  6198.1 1801.08  6203.3 1800.25  6219.0 1807.79
#Mann=15,-1,0
  4664.5     0.1       0  4675.0    0.07       0  4842.6     0.1       0
  4863.1   0.033       0  4982.7   0.033       0  5000.4   0.033       0
  5060.9    0.07       0  5170.3   0.035       0  5272.5    0.07       0
  5359.0   0.035       0  5416.3    0.07       0  5575.4   0.035       0
  5758.6    0.07       0  5793.0   0.035       0  5986.6     0.1       0
Bank Sta=4982.7,5000.4
Exp/Cntr=0.3,0.1

Type RM Length L Ch R = 1,19186,558,558,558
BEGIN DESCRIPTION:
Palmer Creek 33.0
END DESCRIPTION:
XS GIS Cut Line= 3
      1914690.64     13875232.43      1914520.16     13874645.63
      1913895.82     13873458.35
#Sta/Elev= 30
  4340.3 1761.88  4347.6 1761.57  4350.4 1761.48  4523.2 1758.28  4598.3 1757.36
  4618.8 1753.61  4650.0 1742.38  4681.3 1738.48  4776.5 1745.30  4816.6 1744.45
  4850.1 1738.01  4868.7 1732.46  5006.3 1732.28  5006.8 1731.78  5024.0 1732.28
  5024.8 1732.43  5027.5 1732.93  5103.4 1736.88  5312.5 1738.36  5378.6 1749.11
  5662.4 1747.61  5813.8 1750.42  5899.1 1762.20  5940.4 1766.84  5984.5 1778.45
  6111.0 1821.20  6127.1 1824.22  6133.1 1828.43  6155.1 1832.25  6292.8 1880.88
#Mann=11,-1,0
  4340.3   0.035       0  4347.6    0.07       0  4350.4   0.035       0
  4523.2    0.07       0  4850.1   0.033       0  5006.3   0.033       0
  5024.0   0.033       0  5024.8     0.1       0  5027.5   0.035       0
  5662.4    0.07       0  5899.1     0.1       0
Bank Sta=5006.3,5024
Exp/Cntr=0.3,0.1

Type RM Length L Ch R = 1,18628,490,490,490
BEGIN DESCRIPTION:
Palmer Creek 32.0
END DESCRIPTION:
XS GIS Cut Line= 3
      1915075.00     13875325.00      1914575.00     13874125.00
      1913909.61     13873391.42
#Sta/Elev= 30
  3706.5 1775.98  3816.5 1767.87  4023.0 1754.31  4140.9 1752.71  4275.9 1755.75
  4334.8 1753.86  4365.7 1746.95  4371.1 1742.17  4400.4 1738.00  4587.3 1735.07
  4845.9 1732.28  4846.4 1731.78  4863.8 1732.28  4948.4 1732.40  5009.9 1732.67
  5048.7 1739.54  5056.2 1735.59  5062.9 1739.19  5091.3 1737.20  5098.8 1742.94
  5112.9 1744.29  5133.9 1740.17  5155.0 1745.55  5235.5 1747.31  5247.6 1747.28
  5534.9 1758.62  5600.9 1771.19  5891.5 1880.96  5919.9 1888.44  5996.9 1896.14
#Mann=12,-1,0
  3706.5    0.07       0  3816.5   0.035       0  4023.0    0.07       0
  4140.9   0.035       0  4275.9    0.07       0  4587.3   0.033       0
  4845.9    0.05       0  4863.8   0.033       0  4948.4    0.07       0
  5235.5   0.035       0  5247.6    0.07       0  5534.9     0.1       0
Bank Sta=4845.9,4863.8
Exp/Cntr=0.3,0.1

Type RM Length L Ch R = 1,18138,469,469,469
BEGIN DESCRIPTION:
Palmer Creek 31.0
END DESCRIPTION:
XS GIS Cut Line= 3
      1914875.00     13874724.96      1914925.00     13874175.00
      1915225.00     13873825.00
#Sta/Elev= 30
  4447.5 1754.53  4557.9 1749.78  4581.9 1747.19  4628.2 1740.45  4648.3 1739.44
  4819.0 1738.34  4940.9 1733.74  4980.7 1732.19  4981.2 1731.69  4998.6 1732.19
  5035.3 1732.48  5205.5 1733.61  5226.4 1754.99  5240.6 1767.67  5262.6 1778.95
  5283.4 1785.86  5312.0 1790.87  5326.2 1798.43  5332.8 1804.43  5340.5 1808.49
  5347.1 1815.29  5354.8 1820.66  5368.5 1835.84  5382.2 1846.03  5389.9 1849.48
  5405.7 1860.51  5418.4 1872.56  5425.0 1876.21  5432.7 1878.34  5460.7 1879.76
#Mann=7,-1,0
  4447.5    0.07       0  4581.9   0.035       0  4940.9    0.07       0
  4980.7    0.05       0  4998.6    0.07       0  5035.3   0.033       0
  5405.7     0.1       0
Bank Sta=4980.7,4998.6
Exp/Cntr=0.3,0.1

Type RM Length L Ch R = 1,17669,416,416,416
BEGIN DESCRIPTION:
Palmer Creek 30.0
END DESCRIPTION:
XS GIS Cut Line= 3
      1914925.03     13874724.97      1915225.00     13874475.00
      1915325.01     13873974.97
#Sta/Elev= 30
  4609.6 1754.02  4675.2 1751.42  4758.6 1745.75  4857.5 1743.31  4894.0 1743.61
  4957.8 1741.45  4964.3 1737.38  4977.4 1732.47  4977.9 1731.97  4995.4 1732.47
  5057.0 1732.65  5142.8 1732.85  5183.6 1734.04  5234.6 1741.39  5265.2 1746.75
  5275.4 1749.49  5285.6 1755.43  5306.0 1763.27  5326.4 1774.03  5336.6 1782.12
  5377.4 1803.42  5389.2 1812.95  5408.0 1824.83  5418.2 1833.02  5428.4 1837.15
  5438.6 1845.91  5469.2 1857.19  5479.4 1865.15  5489.6 1871.33  5510.0 1872.00
#Mann=6,-1,0
  4609.6    0.07       0  4675.2   0.035       0  4977.4   0.035       0
  4995.4   0.035       0  5057.0   0.033       0  5389.2     0.1       0
Bank Sta=4977.4,4995.4
Exp/Cntr=0.3,0.1

Type RM Length L Ch R = 1,17253,469,469,469
BEGIN DESCRIPTION:
Palmer Creek 29.0
END DESCRIPTION:
XS GIS Cut Line= 3
      1915125.01     13875024.98      1915525.00     13874425.00
      1915375.00     13874024.99
#Sta/Elev= 30
  4273.2 1753.71  4605.2 1744.13  4791.5 1742.09  4814.0 1740.00  4821.5 1736.16
  4836.5 1732.76  4917.3 1732.22  5080.5 1732.12  5081.0 1731.62  5098.5 1732.12
  5143.8 1740.78  5175.0 1753.62  5180.3 1753.49  5205.2 1768.89  5229.2 1777.83
  5235.5 1783.23  5254.5 1791.10  5265.7 1793.54  5290.7 1808.90  5296.0 1809.73
  5314.7 1819.82  5320.9 1825.13  5326.3 1825.90  5345.8 1837.03  5351.2 1838.16
  5357.4 1843.79  5381.4 1854.45  5389.4 1860.10  5406.4 1865.56  5421.5 1867.14
#Mann=5,-1,0
  4273.2   0.035       0  4917.3   0.033       0  5080.5   0.033       0
  5098.5   0.033       0  5254.5     0.1       0
Bank Sta=5080.5,5098.5
Exp/Cntr=0.3,0.1

Type RM Length L Ch R = 1,16784,916,916,916
BEGIN DESCRIPTION:
Palmer Creek 28.0
END DESCRIPTION:
XS GIS Cut Line= 3
      1915274.99     13875175.01      1915875.00     13874575.00
      1915825.00     13874224.99
#Sta/Elev= 30
  4151.1 1756.63  4154.6 1756.63  4165.3 1754.77  4250.1 1750.01  4419.8 1745.08
  4688.5 1740.01  4815.8 1737.08  4900.6 1736.03  4934.5 1736.47  4957.2 1735.69
  4987.1 1732.31  4987.6 1731.81  5004.6 1731.81  5005.1 1732.31  5029.9 1732.50
  5040.0 1733.25  5051.2 1733.40  5110.8 1734.40  5176.4 1733.26  5181.5 1732.64
  5211.8 1732.50  5221.9 1734.58  5242.1 1746.96  5262.3 1758.65  5272.4 1762.26
  5282.5 1767.27  5292.6 1771.00  5302.7 1772.70  5322.9 1775.18  5353.2 1776.30
#Mann=5,-1,0
  4151.1   0.035       0  4934.5     0.1       0  4987.1    0.05       0
  5005.1     0.1       0  5051.2   0.033       0
Bank Sta=4987.1,5005.1
Exp/Cntr=0.3,0.1
