--- Town Creek.prj (project) ---

Proj Title=Town Creek Base Level Engineering
Current Plan=p01
Default Exp/Contr=0.3,0.1
English Units
Geom File=g01
Flow File=f01
Plan File=p01
Y Axis Title=Elevation
X Axis Title(PF)=Main Channel Distance
X Axis Title(XS)=Station
BEGIN DESCRIPTION:
Town Creek
END DESCRIPTION:
DSS Export Rating Curves= 0
DSS Export Rating Curve Sorted= 0
DSS Export Volume Flow Curves= 0
DXF OffsetX= 0
DXF OffsetY= 0
DXF ScaleX= 1
DXF ScaleY= 10

--- Town Creek.p01 (plan) ---

Plan Title=Multiple Run
Short Identifier=Multiple
Geom File=g01
Flow File=f01
Subcritical Flow
K Sum by GR= 0
Std Step Tol= 0.01
Critical Tol= 0.01
Num of Std Step Trials= 20
Max Error Tol= 0.3
Flow Tol Ratio= 0.001
Split Flow NTrial= 30
Split Flow Tol= 0.02
Split Flow Ratio= 0.02
Log Output Level= 0
Friction Slope Method= 1
Unsteady Friction Slope Method= 2
Unsteady Bridges Friction Slope Method= 1
Parabolic Critical Depth
Global Vel Dist=  1 , 1 , 1
Global Log Level= 0
CheckData=True
Encroach Param= -1, 0, 0, 0
BEGIN DESCRIPTION:
Multiple Run
END DESCRIPTION:

--- Town Creek.f01 (steady flow) ---

Flow Title=Multiple
Number of Profiles=7
Profile Names=10-year,25-year,50-year,1pct_min,100-year,1pct_plu,500-year
River Rch & RM= Town Creek,Reach-1,48171
    2328    4154    5966    4133    8247   16454   15579
River Rch & RM= Town Creek,Reach-1,44098
    2484    4439    6381    4422    8823   17605   16684
River Rch & RM= Town Creek,Reach-1,42376
    3738    6813    9926    6963   13892   27718   26921
River Rch & RM= Town Creek,Reach-1,41140
    3825    6974   10162    7128   14222   28376   27558
River Rch & RM= Town Creek,Reach-1,40239
    3956    7212   10508    7368   14700   29331   28467
River Rch & RM= Town Creek,Reach-1,37289
    5434    9993   14648   10324   20599   41101   40292
River Rch & RM= Town Creek,Reach-1,35077
    5624   10341   15154   10675   21300   42499   41622
River Rch & RM= Town Creek,Reach-1,31470
    6554   12114   17816   12590   25120   50121   49393
River Rch & RM= Town Creek,Reach-1,30565
    6641   12271   18042   12745   25429   50737   49962
River Rch & RM= Town Creek,Reach-1,27828
    7030   13011   19152   13542   27019   53910   53187
River Rch & RM= Town Creek,Reach-1,26723
    7061   13053   19198   13561   27058   53988   53162
River Rch & RM= Town Creek,Reach-1,23947
    7173   13248   19472   13744   27423   54716   53794
River Rch & RM= Town Creek,Reach-1,19826
    7201   13295   19537   13787   27508   54886   53934
River Rch & RM= Town Creek,Reach-1,19210
    9791   18266   27032   19197   38303   76426   76050
River Rch & RM= Town Creek,Reach-1,16699
    9826   18321   27105   19242   38392   76602   76167
River Rch & RM= Town Creek,Reach-1,15579
    9840   18329   27098   19222   38352   76523   75970
River Rch & RM= Town Creek,Reach-1,12493
   10616   19793   29279   20777   41456   82715   82172
River Rch & RM= Town Creek,Reach-1,8943
   10559   19643   29013   20554   41011   81828   81020
River Rch & RM= Town Creek,Reach-1,2263
   10749   19996   29534   20921   41743   83287   82448
Boundary for River Rch & Prof#=Town Creek,Reach-1,1
Up Type=0
Dn Type=3
Dn Slope=0.005
Boundary for River Rch & Prof#=Town Creek,Reach-1,2
Up Type=0
Dn Type=3
Dn Slope=0.005
Boundary for River Rch & Prof#=Town Creek,Reach-1,3
Up Type=0
Dn Type=3
Dn Slope=0.005
Boundary for River Rch & Prof#=Town Creek,Reach-1,4
Up Type=0
Dn Type=3
Dn Slope=0.005
Boundary for River Rch & Prof#=Town Creek,Reach-1,5
Up Type=0
Dn Type=3
Dn Slope=0.005
Boundary for River Rch & Prof#=Town Creek,Reach-1,6
Up Type=0
Dn Type=3
Dn Slope=0.005
Boundary for River Rch & Prof#=Town Creek,Reach-1,7
Up Type=0
Dn Type=3
Dn Slope=0.005

--- Town Creek.g01 (geometry) ---

Geom Title=Existing Conditions
Program Version=4.10

River Reach=Town Creek      ,Reach-1
Reach XY= 30
        1926625.       13962675.      1926245.25      13961644.6
      1924715.21     13960964.48       1924266.9     13960028.35
      1923564.89      13960214.7      1923355.24     13959253.97
      1920835.76     13957284.68      1920375.07     13956059.61
      1920621.53      13955376.5       1919726.2      13954614.5
      1920021.39      13953626.5      1918776.22      13952664.5
      1919366.79     13952131.67      1919627.06     13949880.85
       1920273.8     13948864.49      1919728.72     13946826.54
      1921117.69      13946475.1      1920724.57     13945895.18
       1921073.8      13942335.5       1920176.2      13940785.5
      1921971.37      13938473.5       1921474.9      13937504.9
      1921583.03     13934521.65      1922724.49     13933709.79
      1922295.47     13932894.63      1921382.79     13932428.42
      1922267.47     13930925.01      1922111.38     13930211.78
      1921080.82     13929527.31        1921175.       13929075.

Type RM Length L Ch R = 1 ,48171   ,463,463,463
BEGIN DESCRIPTION:
Town Creek 90.0
END DESCRIPTION:
XS GIS Cut Line= 3
      1926824.96     13962475.01        1926575.       13962525.
      1926274.98     13962825.02
#Sta/Elev= 30
  4745.1 1947.37  4816.9 1922.56    4823 1918.09    4835 1913.06  4841.4 1909.07
  4861.8 1899.35  4905.6 1880.42  4911.8 1876.89    4927 1865.42  4930.1 1864.47
  4945.4 1864.68  4972.9 1865.68  4985.2 1862.08  4999.1 1860.54  4999.4 1860.04
  5003.5 1860.54  5005.5 1860.91  5017.6 1868.66  5026.1 1870.44  5115.2 1872.16
  5149.8 1876.27  5180.7 1882.74  5204.9 1889.13  5246.7 1903.34  5268.3 1908.54
  5306.8 1919.92  5344.9 1926.43  5366.2 1932.29  5416.4 1942.44  5424.3 1942.45
#Mann= 5 ,-1 , 0
  4745.1      .1       0  4945.4     .07       0  4999.1     .05       0
  5003.5     .07       0  5180.7      .1       0
Bank Sta=4999.1,5003.5
XS Rating Curve= 0 ,0
Exp/Cntr=0.3,0.1

Type RM Length L Ch R = 1 ,47708   ,420,420,420
BEGIN DESCRIPTION:
Town Creek 89.0
END DESCRIPTION:
XS GIS Cut Line= 3
      1926575.02     13962024.99        1926325.       13962175.
      1926124.99     13962575.02
#Sta/Elev= 30
  4714.1 1955.22  4746.1 1946.79  4823.1 1918.04  4863.1 1894.11  4886.1 1878.38
  4903.6 1868.54  4910.8  1865.7  4924.6 1863.19  4976.3 1864.01    4979 1862.52
    4984 1855.61  5003.2  1853.9  5003.5  1853.4  5007.8  1853.9  5008.9 1855.28
  5015.6 1857.16  5045.8 1859.77  5072.7 1861.31  5099.5    1860  5112.9 1862.65
  5139.7 1865.12  5178.9 1867.23  5200.1 1867.54  5213.5 1869.22  5300.7 1890.85
  5326.5 1899.26  5360.7 1907.07  5374.5 1909.01  5418.1 1918.47  5452.9 1921.93
#Mann= 5 ,-1 , 0
  4714.1      .1       0  4910.8     .07       0  5003.2     .05       0
  5007.8     .07       0  5178.9      .1       0
Bank Sta=5003.2,5007.8
XS Rating Curve= 0 ,0
Exp/Cntr=0.3,0.1

Type RM Length L Ch R = 1 ,47288   ,504,504,504
BEGIN DESCRIPTION:
Town Creek 88.0
END DESCRIPTION:
XS GIS Cut Line= 4
      1926525.03     13961875.01      1926393.34     13961822.34
      1926202.39     13961806.12      1925923.91     13962017.18
#Sta/Elev= 30
  4738.1 1943.23    4772 1935.39    4814 1919.52  4824.7 1913.31  4830.2 1911.36
  4839.9 1905.26  4852.8 1899.82  4880.1 1885.49    4910 1872.85  4932.9 1858.15
  4938.9 1855.44    4948 1853.71  4985.4 1851.75  4990.1 1852.42  5011.1 1851.02
  5011.4 1850.52  5015.7 1851.02  5023.3 1852.03  5032.3 1855.07  5078.9 1855.62
  5097.7 1860.71  5130.8 1862.76  5175.5 1864.47  5199.4    1863  5309.6 1864.04
  5329.5 1865.55  5347.5  1868.6  5361.1  1871.5  5376.3 1874.88    5421 1880.32
#Mann= 6 ,-1 , 0
  4738.1      .1       0  4985.4     .07       0  5011.1     .05       0
  5015.7     .07       0  5347.5      .1       0  5361.1    .035       0
Bank Sta=5011.1,5015.7
XS Rating Curve= 0 ,0
Exp/Cntr=0.3,0.1

Type RM Length L Ch R = 1 ,46784   ,443,443,443
BEGIN DESCRIPTION:
Town Creek 87.0
END DESCRIPTION:
XS GIS Cut Line= 3
      1926074.99     13961225.04        1925975.       13961575.
      1925874.99     13961925.03
#Sta/Elev= 30
  4631.8 1965.84  4643.1 1963.13  4664.9 1954.14  4683.7 1949.01  4727.3 1933.24
  4739.8 1927.13    4771 1918.15    4796 1908.14  4824.1 1894.62    4849 1879.67
    4877 1861.31  4888.2 1855.93  4896.2 1853.87  4925.1  1852.9  4942.6 1849.61
  4962.1 1849.83  5018.2 1844.33  5018.5 1843.83  5023.1 1844.33  5039.4 1850.13
  5064.3 1850.92  5076.8 1855.26    5083 1856.02  5173.7 1855.02  5254.6 1858.67
  5267.1 1861.08  5298.3 1873.69  5323.3 1877.26  5348.4 1878.53  5359.8  1879.3
#Mann= 6 ,-1 , 0
  4631.8      .1       0  4896.2     .07       0  5018.2     .05       0
  5023.1     .07       0  5173.7      .1       0  5348.4    .035       0
Bank Sta=5018.2,5023.1
XS Rating Curve= 0 ,0
Exp/Cntr=0.3,0.1

Type RM Length L Ch R = 1 ,46341   ,474,474,474
BEGIN DESCRIPTION:
Town Creek 86.0
END DESCRIPTION:
XS GIS Cut Line= 3
      1925774.97     13961175.03        1925575.       13961425.
      1925175.02     13961774.99
#Sta/Elev= 30
  4684.7 1939.63  4749.4  1919.5  4762.7  1914.6  4768.6 1910.99  4812.6 1894.51
  4844.3 1880.31    4886 1856.98    4901 1849.47  4912.5 1846.71  4935.5 1846.96
  4947.1 1843.95  4997.6 1841.02    4998 1840.52  5002.5 1841.02  5050.2 1845.36
  5072.4 1845.83    5100 1849.31  5181.8 1848.66  5204.2  1849.9  5219.4 1852.85
  5263.2 1871.19  5275.2 1873.77    5331  1880.8  5354.9  1886.4  5369.1 1887.04
  5396.5 1891.26  5428.4 1893.35  5446.5 1897.72    5534 1909.63  5536.3 1909.41
#Mann= 6 ,-1 , 0
  4684.7      .1       0    4886     .07       0  4997.6     .05       0
  5002.5     .07       0  5181.8    .035       0    5534      .1       0
Bank Sta=4997.6,5002.5
XS Rating Curve= 0 ,0
Exp/Cntr=0.3,0.1

Type RM Length L Ch R = 1 ,45867   ,444,444,444
BEGIN DESCRIPTION:
Town Creek 85.0
END DESCRIPTION:
XS GIS Cut Line= 3
      1925475.03     13960824.97        1925175.       13961225.
        1925175.     13961324.96
#Sta/Elev= 30
  4504.5 1942.74  4515.7 1939.16  4541.9 1933.48  4553.2 1928.76  4583.2 1922.04
  4598.2 1916.29  4624.4 1908.62  4650.7 1897.03  4665.7 1888.49  4673.2 1882.73
  4703.2 1867.21  4733.2 1854.65  4748.2 1851.74  4763.2 1850.19    4897 1847.93
    4927 1839.19  4939.4 1837.57  4946.9  1838.8  4958.2 1837.41  4973.2 1838.01
  4985.7 1833.25  4986.1 1832.75  4990.7 1833.25  4991.8 1834.66  5003.2 1840.95
  5036.5 1845.24  5057.5  1849.5    5068 1854.72  5078.5 1858.47  5104.5 1860.64
#Mann= 3 ,-1 , 0
  4504.5      .1       0  4985.7     .05       0  4990.7      .1       0
Bank Sta=4985.7,4990.7
XS Rating Curve= 0 ,0
Exp/Cntr=0.3,0.1

Type RM Length L Ch R = 1 ,45423   ,448,448,448
BEGIN DESCRIPTION:
Town Creek 84.0
END DESCRIPTION:
XS GIS Cut Line= 3
      1925225.02     13960674.99        1924825.       13960975.
      1924425.01     13961374.99
#Sta/Elev= 30
  4495.6  1924.3  4515.2 1921.16  4529.9 1916.31  4559.9 1910.69  4615.5 1894.93
  4664.9 1879.66  4691.2 1869.21  4728.7 1856.58  4751.2 1851.74  4762.6 1847.56
  4805.5 1845.25  4938.7 1843.83  4994.9 1836.25    5004 1832.72  5016.4 1829.97
    5047 1829.64  5047.5 1829.14    5053 1829.64  5054.9 1832.48  5076.1 1839.28
  5096.7 1839.15  5114.3 1843.99    5148 1845.58    5284  1851.2  5373.1 1852.56
  5391.9 1853.98  5436.1  1861.6  5491.9 1875.52  5537.9 1889.68  5561.3 1893.84
#Mann= 5 ,-1 , 0
  4495.6      .1       0  4762.6     .07       0    5047     .05       0
    5053     .07       0    5148      .1       0
Bank Sta=5047,5053
XS Rating Curve= 0 ,0
Exp/Cntr=0.3,0.1

Type RM Length L Ch R = 1 ,44975   ,431,431,431
BEGIN DESCRIPTION:
Town Creek 83.0
END DESCRIPTION:
XS GIS Cut Line= 3
      1924874.99     13960475.01        1924475.       13960725.
        1924075.       13960925.
#Sta/Elev= 30
  4532.7 1859.26  4580.4 1855.96  4626.2 1851.15  4638.2 1851.61  4665.3 1848.52
  4683.5    1848  4739.6 1836.83  4813.6 1835.95  4858.9  1833.7  4879.1 1834.99
  4905.9 1834.27    4920 1833.37  4932.5 1830.63  4942.2 1831.59  4962.5 1827.88
  4973.1 1828.31  4993.7 1824.72  4994.2 1824.22  4999.7 1824.72    5015 1830.79
  5031.7 1839.41  5088.1 1841.63  5113.7 1842.65  5195.5 1852.68  5246.4 1862.37
  5276.6 1870.38  5323.5 1887.86  5350.4 1896.51    5404 1919.01  5451.6 1936.55
#Mann= 5 ,-1 , 0
  4532.7      .1       0  4626.2     .07       0  4993.7     .05       0
  4999.7     .07       0  5088.1      .1       0
Bank Sta=4993.7,4999.7
XS Rating Curve= 0 ,0
Exp/Cntr=0.3,0.1

Type RM Length L Ch R = 1 ,44544   ,446,446,446
BEGIN DESCRIPTION:
Town Creek 82.0
END DESCRIPTION:
XS GIS Cut Line= 3
      1924775.01     13959924.99        1924375.       13960325.
      1923974.99     13960725.01
#Sta/Elev= 30
  4434.8 1914.13  4486.4    1900  4528.8 1891.12  4594.2 1870.62  4621.4 1861.37
  4659.5 1841.07  4670.5 1838.38  4757.1 1836.26  4769.9 1833.83  4779.1 1829.59
  4783.4 1833.93  4789.3 1835.18  4850.2 1833.24  4901.8 1828.67  4933.6 1829.19
  4978.5 1823.61  5013.5 1822.42    5014 1821.92    5020 1822.42  5037.9  1825.5
  5054.1 1832.99  5063.4 1835.02  5183.9 1837.31  5240.8 1837.77  5287.5 1840.28
  5376.5 1857.46  5397.8 1863.98    5419 1873.83  5442.7 1881.11  5566.2 1938.46
#Mann= 5 ,-1 , 0
  4434.8      .1       0  4850.2     .07       0  5013.5     .05       0
    5020     .07       0  5183.9      .1       0
Bank Sta=5013.5,5020
XS Rating Curve= 0 ,0
Exp/Cntr=0.3,0.1

Type RM Length L Ch R = 1 ,44098   ,693,693,693
BEGIN DESCRIPTION:
Town Creek 81.0
END DESCRIPTION:
XS GIS Cut Line= 3
        1924175.       13959875.        1924175.       13959975.
        1923875.       13960375.
#Sta/Elev= 30
  4895.3 1843.33  4930.2  1841.5  4948.2 1841.13  4957.2 1841.84  4966.2 1840.55
  4975.2 1834.57  4984.2 1827.89  4987.2 1824.56  4993.2 1820.68  4998.4 1818.72
  5003.6  1818.1  5004.1  1817.6  5010.3  1818.1  5017.7 1819.95  5037.7 1821.94
  5079.8 1823.38  5127.7 1826.74  5162.3 1827.44  5201.1 1827.81  5366.1 1826.79
  5381.1 1827.84  5392.7 1830.39  5401.4 1833.51  5405.6 1834.07  5412.7 1837.15
  5423.9 1842.51  5431.4 1847.16  5450.2 1857.11  5463.4  1863.2  5495.3 1879.51
#Mann= 4 ,-1 , 0
  4895.3     .07       0  5003.6     .05       0  5010.3     .07       0
  5162.3      .1       0
Bank Sta=5003.6,5010.3
XS Rating Curve= 0 ,0
Exp/Cntr=0.3,0.1

Type RM Length L Ch R = 1 ,43405   ,470,470,470
BEGIN DESCRIPTION:
Town Creek 80.0
END DESCRIPTION:
XS GIS Cut Line= 4
      1924095.37     13959591.63       1923729.8      13959880.3
      1923620.06     13960157.22      1923705.38     13960439.42
#Sta/Elev= 30
  4164.7  1852.4  4174.6 1852.08  4184.5 1848.52  4242.4 1840.08  4312.3 1834.77
  4435.7 1831.61    4475 1831.53  4670.6 1825.26    4714 1823.18  4823.7 1824.33
  4868.9 1816.63  4917.1 1817.16  4960.6 1817.65    4995 1813.28    5002 1811.85
  5002.5 1811.35  5008.7 1811.85  5009.5 1815.09  5014.8 1818.57  5027.3 1822.07
  5036.7 1828.35  5049.2 1839.06  5061.8 1846.84    5068 1852.69  5092.4 1868.33
  5099.4 1875.31  5106.9  1885.1  5111.9  1893.2  5162.1 1903.36  5223.2 1912.92
#Mann= 9 ,-1 , 0
  4164.7      .1       0  4174.6    .035       0  4242.4      .1       0
  4435.7     .07       0  4670.6      .1       0  4917.1     .07       0
    4995      .1       0    5002     .05       0  5008.7      .1       0
Bank Sta=5002,5008.7
XS Rating Curve= 0 ,0
Exp/Cntr=0.3,0.1

Type RM Length L Ch R = 1 ,42935   ,166,166,166
BEGIN DESCRIPTION:
Town Creek 79.0
END DESCRIPTION:
XS GIS Cut Line= 3
      1924204.17     13959509.78      1923534.84     13959853.34
      1922836.94     13959845.58
#Sta/Elev= 30
  4187.8 1892.54  4251.5 1873.71  4288.8 1859.84  4359.9 1846.69  4387.9 1842.81
  4497.6 1833.24  4816.8 1825.11  4878.7 1820.48  4925.9 1813.11  5011.1 1811.05
  5011.6 1810.55  5017.8 1811.05  5026.5 1813.58  5053.5 1834.53  5087.7 1830.04
  5110.5 1817.44  5127.3 1817.39  5134.5 1817.42  5146.5 1824.33  5161.5 1825.79
  5221.8 1821.16  5278.5 1820.17  5300.2 1814.07  5305.5 1812.49  5404.5 1812.22
  5455.5 1840.31  5503.5 1854.29  5554.5 1878.97  5575.5 1891.47  5638.1 1910.94
#Mann= 7 ,-1 , 0
  4187.8      .1       0  4359.9    .035       0  4387.9      .1       0
  5011.1     .05       0  5017.8      .1       0  5127.3    .035       0
  5300.2      .1       0
Bank Sta=5011.1,5017.8
XS Rating Curve= 0 ,0
Exp/Cntr=0.3,0.1

Type RM Length L Ch R = 1 ,42769   ,393,393,393
BEGIN DESCRIPTION:
Town Creek 78.0
END DESCRIPTION:
XS GIS Cut Line= 3
      1923930.85     13959543.15      1923483.63     13959688.35
      1923075.02       13959625.
#Sta/Elev= 30
  4521.1 1838.61  4607.5 1833.34  4668.6 1829.55  4750.2 1827.16  4821.2 1827.79
  4873.6 1825.76    4902  1822.4  4956.9  1810.9  4999.5 1812.79  5014.5 1809.14
  5025.1 1809.19    5058 1819.66  5080.3 1820.36    5096 1818.61  5102.7 1812.69
  5108.8 1811.85    5130 1817.55    5146 1818.75  5165.7 1817.87  5177.5 1812.53
  5214.3 1811.04  5236.3 1812.65  5276.1 1810.38  5295.1 1808.44  5295.6 1807.94
  5301.8 1808.44  5311.6 1810.98  5327.3 1821.59  5335.2 1823.92  5404.8 1826.76
#Mann= 6 ,-1 , 0
  4521.1      .1       0  4607.5     .07       0  4750.2      .1       0
  5276.1    .035       0  5295.1     .05       0  5301.8    .035       0
Bank Sta=5295.1,5301.8
XS Rating Curve= 0 ,0
Exp/Cntr=0.3,0.1

Type RM Length L Ch R = 1 ,42376   ,283,283,283
BEGIN DESCRIPTION:
Mapping XS 91e08b51
END DESCRIPTION:
XS GIS Cut Line= 3
      1923742.28     13959127.95      1923285.86     13959377.15
      1922978.97     13959629.28
#Sta/Elev= 30
  4587.5 1854.58    4618 1844.03  4664.7 1834.51  4706.8 1827.15  4737.3 1825.03
    4806 1822.97  4867.5 1822.94  4877.7 1823.37  4885.8 1822.29  4918.8 1821.79
  4946.9 1811.56  4952.9 1809.09    4998 1808.05  5002.1 1807.82  5002.6 1807.32
  5013.1 1807.82  5013.2 1808.94  5048.6 1808.68  5079.4 1814.85  5091.9 1815.48
  5195.9 1817.05  5261.9 1819.68  5300.2 1822.28  5304.7  1821.9  5378.4 1825.44
  5402.4 1828.09  5421.1  1827.9  5441.8 1830.38    5460  1834.9  5504.7 1854.41
#Mann= 11 ,-1 , 0
  4587.5      .1       0  4664.7     .07       0  4737.3    .035       0
  4867.5      .1       0  4946.9     .07       0    4998      .1       0
  5002.1     .05       0  5013.1      .1       0  5091.9     .07       0
  5300.2    .035       0  5441.8      .1       0
Bank Sta=5002.1,5013.1
XS Rating Curve= 0 ,0
Exp/Cntr=0.3,0.1

Type RM Length L Ch R = 1 ,42093   ,489,489,489
BEGIN DESCRIPTION:
Town Creek 77.0
END DESCRIPTION:
XS GIS Cut Line= 3
      1923625.04     13958874.97      1923186.72     13959236.04
      1922874.98     13959675.03
#Sta/Elev= 30
    4431  1869.2  4543.7 1835.71  4581.9 1824.64  4685.7 1820.84  4729.6 1820.14
  4756.8 1817.45  4770.6  1812.7  4790.8 1808.86  4841.4 1808.11  4867.7 1809.25
    4889 1808.15  4960.9 1809.29  4974.1 1809.04  4977.5 1807.43    4978 1806.93
  4988.5 1807.43  4993.2 1808.05  4997.8 1810.59  5019.6 1814.61  5100.5  1816.1
  5178.5 1820.49    5241 1824.45  5284.5 1829.34  5303.2  1828.8  5311.6 1831.08
    5344 1834.86  5365.3 1840.15  5398.6 1854.15  5451.5 1870.65  5537.3 1901.69
#Mann= 9 ,-1 , 0
    4431      .1       0  4543.7    .035       0  4685.7      .1       0
  4867.7    .035       0  4960.9     .07       0  4977.5     .05       0
  4988.5     .07       0  5178.5    .035       0    5344      .1       0
Bank Sta=4977.5,4988.5
XS Rating Curve= 0 ,0
Exp/Cntr=0.3,0.1

Type RM Length L Ch R = 1 ,41604   ,464,464,464
BEGIN DESCRIPTION:
Town Creek 76.0
END DESCRIPTION:
XS GIS Cut Line= 3
      1923501.35      13958721.7      1922962.63     13958961.83
        1922675.       13959475.
#Sta/Elev= 30
    4373 1839.51  4411.1 1833.76  4496.5 1828.98  4509.6 1829.48  4535.2 1827.01
  4742.1 1822.52  4765.8 1822.33  4775.7 1820.66  4782.3 1818.65  4793.5 1810.77
  4864.4  1807.9  4876.9    1809    4904 1807.22  4904.5 1806.72    4915 1807.22
  5038.6  1807.8  5055.3 1809.75  5086.7 1815.73    5128 1818.29  5203.6 1826.89
  5245.2 1837.54  5276.8 1838.15  5310.3 1838.97  5312.7 1841.01  5317.8  1848.9
  5341.2 1858.44  5387.6 1873.26  5461.6 1893.57  5533.6 1910.79  5551.1 1913.22
#Mann= 10 ,-1 , 0
    4373      .1       0  4411.1    .035       0  4535.2      .1       0
  4742.1    .033       0  4876.9     .07       0    4904     .05       0
    4915     .07       0  5055.3    .035       0  5276.8     .07       0
  5387.6      .1       0
Bank Sta=4904,4915
XS Rating Curve= 0 ,0
Exp/Cntr=0.3,0.1

Type RM Length L Ch R = 1 ,41140   ,276,276,276
BEGIN DESCRIPTION:
Town Creek 75.0
END DESCRIPTION:
XS GIS Cut Line= 3
      1923078.32     13958355.47       1922738.7     13958657.27
        1922425.       13959175.
#Sta/Elev= 30
  4486.7 1836.53  4563.7 1831.52  4708.7 1826.13  4802.5 1825.48  4830.2 1825.07
  4882.4 1820.92  4907.4 1817.49    4921 1813.89    4941 1809.89  4974.5 1809.48
  4982.9  1807.9  4983.4  1807.4  4994.3  1807.9  5038.3 1808.02    5117 1808.14
  5121.9 1808.39  5129.1 1811.57  5139.4 1815.12  5150.6    1816  5311.3 1821.48
  5349.9 1825.87  5367.4 1831.19  5376.5 1831.14  5388.4 1831.06    5406 1835.79
  5441.1  1850.6  5455.1 1853.17  5489.3 1866.09  5539.6 1882.69  5546.4 1884.85
#Mann= 11 ,-1 , 0
  4486.7    .035       0  4563.7     .07       0  4802.5      .1       0
    4921    .033       0  4982.9    .033       0  4994.3    .033       0
  5038.3     .07       0  5129.1    .035       0  5376.5      .1       0
  5489.3     .07       0  5539.6      .1       0
Bank Sta=4982.9,4994.3
XS Rating Curve= 0 ,0
Exp/Cntr=0.3,0.1

Type RM Length L Ch R = 1 ,40864   ,625,625,625
BEGIN DESCRIPTION:
Town Creek 74.0
END DESCRIPTION:
XS GIS Cut Line= 3
      1922774.95     13958475.01        1922525.       13958525.
        1922225.       13958925.
#Sta/Elev= 30
  4749.8 1823.95    4779  1823.5  4781.8 1822.91    4813  1822.3  4858.3 1820.19
  4873.6 1820.15  4880.2 1819.13  4903.4 1817.92  4925.6 1815.94    4947 1809.78
  4956.2 1808.41    4999 1807.95  4999.5 1807.45  5009.9 1807.45  5010.4 1807.95
  5141.1 1809.48  5149.6 1809.66  5155.5 1812.41  5160.8 1813.26  5175.5 1812.96
  5194.6 1811.49  5214.3 1811.04  5261.1 1813.41  5307.1 1815.13  5381.2 1819.15
  5430.7 1820.99  5453.3 1823.07  5472.1 1826.66  5480.1 1827.65  5504.7 1828.19
#Mann= 9 ,-1 , 0
  4749.8     .07       0    4779      .1       0  4880.2    .033       0
    4999    .033       0  5010.4    .033       0  5141.1      .1       0
  5261.1    .035       0  5381.2     .07       0  5480.1    .035       0
Bank Sta=4999,5010.4
XS Rating Curve= 0 ,0
Exp/Cntr=0.3,0.1

Type RM Length L Ch R = 1 ,40239   ,138,138,138
BEGIN DESCRIPTION:
Town Creek 73.0
END DESCRIPTION:
XS GIS Cut Line= 3
      1922725.01     13957974.99       1922346.5     13958187.15
      1921925.03     13958724.96
#Sta/Elev= 30
  4560.2  1875.5  4623.1 1856.68  4639.8 1852.45  4659.3 1846.21  4670.5 1841.78
  4676.5 1840.32  4688.9 1833.89  4707.5 1833.95  4724.7 1829.36    4735 1829.15
  4752.2 1827.35  4788.1 1826.19  4854.5 1823.67  4882.9 1823.28  4923.4 1810.75
  4958.3 1809.71  4974.1 1807.98  5038.8 1807.86  5039.3 1807.36    5050 1807.36
  5050.5 1807.86  5178.6 1808.12  5292.4  1808.1  5464.2 1814.39    5526 1817.99
  5540.1 1819.59  5544.4 1821.16  5559.2 1824.89    5582 1829.23  5677.4 1833.86
#Mann= 8 ,-1 , 0
  4560.2      .1       0  4623.1    .035       0  4788.1     .07       0
  4958.3    .033       0  5038.8    .033       0  5050.5    .033       0
  5178.6    .035       0  5544.4     .07       0
Bank Sta=5038.8,5050.5
XS Rating Curve= 0 ,0
Exp/Cntr=0.3,0.1

Type RM Length L Ch R = 1 ,40101   ,97,97,97
BEGIN DESCRIPTION:
Town Creek 72.0
END DESCRIPTION:
XS GIS Cut Line= 3
      1922721.96     13957890.27      1922196.85     13958182.49
        1921825.       13958525.
#Sta/Elev= 30
  4413.7 1906.25  4482.9 1885.65  4563.5  1857.6  4610.1 1843.42  4625.5 1837.06
  4646.5 1837.39  4661.8 1834.77  4734.4 1830.76  4803.7 1826.12  4811.3  1823.5
  4821.6 1821.99  4834.5 1817.74    4853 1814.96  4883.6 1816.66  4890.1 1816.25
  4897.1 1813.84  4908.6  1808.1  4926.3 1807.97  5004.6 1807.77  5005.1 1807.27
  5016.3 1807.77  5060.3 1808.09  5197.2 1807.88  5246.2 1809.09  5279.1 1808.36
  5401.2 1811.16    5446 1814.17  5470.2 1819.83  5500.8 1823.59  5520.2 1825.21
#Mann= 8 ,-1 , 0
  4413.7      .1       0  4563.5    .035       0  4734.4     .07       0
  4926.3    .033       0  5004.6    .033       0  5016.3    .033       0
  5060.3    .035       0  5500.8     .07       0
Bank Sta=5004.6,5016.3
XS Rating Curve= 0 ,0
Exp/Cntr=0.3,0.1

Type RM Length L Ch R = 1 ,40004   ,129,129,129
BEGIN DESCRIPTION:
Town Creek 72.1
END DESCRIPTION:
XS GIS Cut Line= 5
      1922791.01     13957569.54      1922328.78     13957973.18
      1922148.66     13958114.24       1922072.7     13958179.34
       1921760.2     13958489.68
#Sta/Elev= 30
  4130.3 1890.29  4165.4 1885.41  4203.8 1872.92  4253.1 1862.19    4262 1864.33
  4285.9 1865.53  4308.7 1860.32  4340.7 1858.79  4360.6 1855.77  4454.7 1855.69
  4472.5 1857.94  4486.6 1854.38  4518.5 1841.23  4555.5 1836.19  4574.6 1835.84
  4614.3 1843.73  4640.5  1843.5  4804.5 1825.81  4881.4 1819.39  4960.2 1817.09
  5148.8 1816.02  5222.4 1808.54  5257.9 1807.33  5258.4 1806.83  5269.6 1807.33
  5290.2 1807.74  5378.8 1811.33    5400 1813.45    5438 1820.52  5513.2 1824.07
#Mann= 5 ,-1 , 0
  4130.3      .1       0  4555.5    .035       0  5257.9    .035       0
  5269.6    .035       0  5290.2     .07       0
Bank Sta=5257.9,5269.6
XS Rating Curve= 0 ,0
Exp/Cntr=0.3,0.1

Type RM Length L Ch R = 1 ,39875   ,317,317,317
BEGIN DESCRIPTION:
Town Creek 71.1
END DESCRIPTION:
XS GIS Cut Line= 3
      1922244.95     13957568.84      1922125.04     13957974.05
      1921773.07     13958319.14
#Sta/Elev= 30
  4470.6 1933.62  4556.2 1911.84  4650.3 1883.04  4687.6 1870.65  4709.5 1855.74
  4718.9  1852.2  4734.5 1849.63  4765.8 1848.42  4805.7 1838.63  4872.2 1821.69
  4887.8 1819.14    4903 1814.46  4911.5 1805.92  4924.4 1797.27  4931.6 1794.02
  4973.9 1791.55  4991.5 1790.51    4992 1790.01  5003.2 1790.51  5014.3 1791.82
  5048.7 1799.86  5164.4 1799.25  5172.9 1803.27  5185.8 1805.97  5190.1 1810.23
  5194.4 1810.81  5250.1 1806.15  5292.4 1806.91  5308.4 1806.15  5386.1 1814.21
#Mann= 7 ,-1 , 0
  4470.6      .1       0  4650.3    .035       0  4805.7     .07       0
  4973.9    .035       0  4991.5    .035       0  5003.2    .035       0
  5292.4     .07       0
#XS Ineff= 2 , 0
                          5196.2         1810.66
Permanent Ineff=
       F       F
Bank Sta=4991.5,5003.2
XS Rating Curve= 0 ,0
Exp/Cntr=0.3,0.1

Type RM Length L Ch R = 1 ,39558   ,442,442,442
BEGIN DESCRIPTION:
Town Creek 71.0
END DESCRIPTION:
XS GIS Cut Line= 3
      1921925.01     13957624.98        1921825.       13957875.
      1921625.02     13958124.97
#Sta/Elev= 30
  4734.9 1922.96  4762.8 1912.63  4791.9 1897.55  4798.4 1892.88  4804.8  1885.3
  4808.1 1883.81  4815.2 1877.89  4824.2 1872.04  4843.6 1861.79  4849.3 1854.69
  4859.8 1845.68  4875.9 1835.13  4882.4 1831.94  4888.8 1833.23  4908.2 1833.16
  4915.1 1831.28  4930.8  1818.8  4959.9 1800.96  4972.8 1791.69  4980.7 1788.57
  4981.2 1788.07  4992.4 1788.57  5115.7 1792.58    5156 1794.21  5182.1 1797.14
    5209 1801.73    5232 1802.71  5243.4 1801.87  5291.5  1809.3  5324.3 1811.29
#Mann= 6 ,-1 , 0
  4734.9      .1       0  4849.3    .035       0  4915.1     .07       0
  4980.7     .05       0  4992.4     .07       0  5115.7    .035       0
Bank Sta=4980.7,4992.4
XS Rating Curve= 0 ,0
Exp/Cntr=0.3,0.1

Type RM Length L Ch R = 1 ,39116   ,436,436,436
BEGIN DESCRIPTION:
Town Creek 70.0
END DESCRIPTION:
XS GIS Cut Line= 3
      1921725.03     13957474.98        1921475.       13957675.
      1921375.04     13957974.88
#Sta/Elev= 30
  4671.6 1926.65  4700.4 1915.01  4719.6  1904.1  4723.5 1900.82  4737.1 1881.75
  4741.9 1876.77    4753 1868.64  4770.7 1859.44  4776.5 1854.55  4787.8 1847.93
  4811.8 1836.12  4834.9 1822.28  4877.1 1807.05    4904  1807.1    4951 1798.64
  4965.5 1792.27    4975 1789.82  5001.2 1788.46    5065 1788.57  5077.5 1788.32
    5078 1787.82  5089.4 1788.32  5089.7  1789.8  5115.4 1791.91  5137.2 1796.75
  5160.5 1799.48  5200.4 1803.18    5222 1803.59  5282.6 1808.43  5307.9 1809.01
#Mann= 7 ,-1 , 0
  4671.6      .1       0  4787.8    .035       0    4951     .07       0
    5065     .07       0  5077.5     .05       0  5089.4     .07       0
    5222     .07       0
Bank Sta=5077.5,5089.4
XS Rating Curve= 0 ,0
Exp/Cntr=0.3,0.1

Type RM Length L Ch R = 1 ,38680   ,455,455,455
BEGIN DESCRIPTION:
Town Creek 69.0
END DESCRIPTION:
XS GIS Cut Line= 3
      1921524.97     13957375.01        1921125.       13957525.
      1921024.99     13957725.02
#Sta/Elev= 30
    4577 1857.15  4577.4 1857.01  4593.8 1849.52    4602 1847.32  4625.4    1837
  4637.3 1833.08  4659.7  1822.7  4685.3 1816.66  4691.7 1815.76  4701.3 1816.32
  4707.9 1814.26  4717.4 1811.86  4746.2 1808.75  4752.6 1807.16  4765.4 1801.77
  4773.2 1800.13  4839.1 1796.88  4909.9 1789.88  4931.2 1788.82  4961.3 1788.09
  4961.8 1787.59  4973.3 1788.09  5044.3 1788.59  5057.7 1793.51  5067.8 1796.06
  5136.9 1799.22  5151.6 1801.56  5195.2 1805.47  5218.7 1806.65  5227.8 1805.91
#Mann= 7 ,-1 , 0
    4577      .1       0  4577.4     .07       0  4707.9    .035       0
  4931.2      .1       0  4961.3     .05       0  4973.3      .1       0
  5136.9    .035       0
Bank Sta=4961.3,4973.3
XS Rating Curve= 0 ,0
Exp/Cntr=0.3,0.1

Type RM Length L Ch R = 1 ,38225   ,85,85,85
BEGIN DESCRIPTION:
Town Creek 68.0
END DESCRIPTION:
XS GIS Cut Line= 4
      1921224.99     13956875.01        1920825.       13957275.
       1920702.5     13957502.81      1920739.88      13957836.8
#Sta/Elev= 30
  4439.1 1828.74  4509.7 1809.28  4516.3 1808.47  4540.1 1803.85  4574.1 1800.07
  4605.5  1797.9  4680.5 1795.56  4747.6 1794.93  4786.2 1789.23  4809.9 1787.63
  4810.4 1787.13  4821.9 1787.63  4823.6 1788.64  4841.4 1789.27  4928.3 1788.18
  5000.4 1788.02  5029.6  1788.2  5037.5 1789.91  5060.3 1792.37  5094.4 1794.55
  5142.1 1795.44  5162.5 1797.11  5180.3 1799.88    5200 1801.14  5258.2  1802.6
  5294.4 1802.85  5389.5 1805.25  5433.6 1807.54  5485.3 1806.67  5599.5 1808.93
#Mann= 10 ,-1 , 0
  4439.1      .1       0  4516.3     .07       0  4680.5     .07       0
  4809.9     .05       0  4821.9     .07       0  4928.3     .07       0
  5000.4    .035       0  5258.2     .07       0  5294.4    .035       0
  5389.5     .07       0
Bank Sta=4809.9,4821.9
XS Rating Curve= 0 ,0
Exp/Cntr=0.3,0.1

Type RM Length L Ch R = 1 ,38140   ,395,395,395
BEGIN DESCRIPTION:
Town Creek 68.1
END DESCRIPTION:
XS GIS Cut Line= 4
      1921325.69     13956698.79      1920879.69     13957119.83
      1920746.23     13957241.36      1920656.15     13957508.33
#Sta/Elev= 30
  4273.5 1877.79  4291.6 1871.67  4299.8 1869.92  4320.5 1861.66  4357.9 1849.15
  4410.9 1834.98    4469 1822.07    4523 1807.67  4555.2 1801.34  4592.7 1797.45
  4668.4  1794.7  4757.8  1794.2  4774.3 1792.05  4786.4  1788.4  4797.2  1787.5
  4815.4 1786.31  4815.9 1785.81  4827.4 1786.31  4852.7 1787.31  4877.4 1795.14
  4893.8 1796.31  5038.5 1796.71  5069.5 1794.84  5100.6 1791.22  5141.8 1794.07
  5170.3 1794.05  5208.3 1795.62  5236.8 1799.51  5293.8  1803.8  5349.1 1803.66
#Mann= 5 ,-1 , 0
  4273.5      .1       0    4523     .07       0  4797.2     .07       0
  4815.4     .05       0  4827.4     .07       0
#XS Ineff= 2 , 0
                          4904.9         1796.57
Permanent Ineff=
       F       F
Bank Sta=4815.4,4827.4
XS Rating Curve= 0 ,0
Exp/Cntr=0.3,0.1

Type RM Length L Ch R = 1 ,37745   ,456,456,456
BEGIN DESCRIPTION:
Town Creek 67.0
END DESCRIPTION:
XS GIS Cut Line= 4
      1921075.01     13956474.99        1920675.       13956875.
      1920548.65      13957051.2      1920683.41     13957862.57
#Sta/Elev= 30
  4434.3  1826.4  4476.5 1812.38  4534.5 1795.94  4564.7  1791.7  4751.7 1788.24
    4850 1788.06  4871.2 1789.24  4891.8 1787.84  4908.7 1788.31  4942.7 1784.97
    4956 1776.86    4990 1777.57  5007.4 1776.07  5007.9 1775.57  5019.4 1776.07
  5039.3 1778.67  5079.9 1779.89  5113.1 1777.46  5136.4 1785.02  5178.6 1788.48
  5439.9 1794.67    5624 1803.46  5687.9 1804.18  5705.4 1803.06  5761.2 1799.47
  5812.8 1799.94  5833.9 1800.82    5865 1804.97  5906.8 1807.99  6039.3 1809.67
#Mann= 6 ,-1 , 0
  4434.3      .1       0  4476.5     .07       0  5007.4     .05       0
  5019.4     .07       0  5178.6    .035       0  5705.4     .07       0
Bank Sta=5007.4,5019.4
XS Rating Curve= 0 ,0
Exp/Cntr=0.3,0.1

Type RM Length L Ch R = 1 ,37289   ,482,482,482
BEGIN DESCRIPTION:
Town Creek 66.0
END DESCRIPTION:
XS GIS Cut Line= 3
      1921075.04     13956374.99        1920475.       13956525.
      1919874.97     13956725.01
#Sta/Elev= 30
  4381.5 1834.97  4424.8 1816.15  4449.2 1805.59    4477 1796.59  4492.4 1792.55
  4514.7 1790.46  4633.4 1786.83  4770.8 1787.22  4891.4 1781.61  4976.2  1771.6
  4976.7  1771.1  4992.1  1771.6  5015.4 1772.26  5034.4 1775.47  5059.7  1787.2
  5076.5 1786.98  5116.6 1782.45  5213.4 1777.86  5293.6 1784.59  5312.7  1789.3
  5337.9 1788.11  5366.4 1791.29  5425.9 1790.97    5431 1791.09  5472.1 1791.55
  5502.2 1799.25  5530.7 1803.92  5578.1 1803.39  5590.8 1808.88  5632.5 1816.24
#Mann= 8 ,-1 , 0
  4381.5      .1       0  4424.8     .07       0  4976.2     .05       0
  4992.1     .07       0  5076.5      .1       0  5213.4    .035       0
  5425.9     .07       0    5431    .035       0
Bank Sta=4976.2,4992.1
XS Rating Curve= 0 ,0
Exp/Cntr=0.3,0.1

Type RM Length L Ch R = 1 ,36807   ,515,515,515
BEGIN DESCRIPTION:
Town Creek 65.0
END DESCRIPTION:
XS GIS Cut Line= 3
      1920974.99       13955925.        1920375.       13956075.
      1919774.97     13956475.02
#Sta/Elev= 30
  4385.4 1798.22  4458.2 1789.46  4507.6 1786.04    4580 1783.86  4810.7 1780.51
  4850.9 1774.07  4875.8  1773.2  4959.1 1771.64  4967.4 1769.69  4967.9 1769.19
  4983.3 1769.69    4990  1771.5  5024.5  1771.6  5063.9 1773.81  5110.3 1775.82
  5145.6 1772.67  5193.3 1773.13  5222.1  1784.6  5229.3    1786  5387.8 1787.03
  5449.2 1787.97  5510.5  1794.4    5561 1795.18  5575.4 1799.68    5602 1802.55
  5683.6 1815.46  5694.4 1818.83  5705.8 1825.79  5716.1 1828.07    5725 1828.12
#Mann= 9 ,-1 , 0
  4385.4      .1       0    4580     .07       0  4875.8      .1       0
  4967.4     .05       0  4983.3      .1       0  5024.5     .07       0
  5063.9      .1       0  5145.6     .07       0  5387.8    .035       0
Bank Sta=4967.4,4983.3
XS Rating Curve= 0 ,0
Exp/Cntr=0.3,0.1

Type RM Length L Ch R = 1 ,36292   ,338,338,338
BEGIN DESCRIPTION:
Mapping XS 7d0163ca
END DESCRIPTION:
XS GIS Cut Line= 3
      1921073.12     13955553.35      1920543.79     13955633.13
      1919611.91     13956077.69
#Sta/Elev= 30
  4496.3 1895.03  4503.1 1890.39  4512.2 1880.59  4524.3 1872.25  4539.5 1863.21
  4563.8  1853.1    4582 1840.46  4629.9 1823.84    4673 1801.35    4692 1793.04
  4717.9 1783.39  4733.7  1781.1  4882.3 1776.16  4933.9 1772.16  4952.1 1768.31
  4993.4 1767.31  4993.9 1766.81  5009.4 1767.31  5044.2 1768.59  5075.1 1776.08
  5136.5 1780.58  5224.9 1781.06  5335.5 1782.34    5439 1782.92  5551.5 1782.69
  5668.3 1785.18  5907.1 1793.68  5998.2 1798.24  6042.1 1804.34  6064.1 1810.56
#Mann= 10 ,-1 , 0
  4496.3      .1       0    4692     .07       0  4993.4     .05       0
  5009.4     .07       0  5136.5    .035       0  5224.9     .07       0
  5335.5    .035       0    5439     .07       0  5668.3    .035       0
  5907.1      .1       0
Bank Sta=4993.4,5009.4
XS Rating Curve= 0 ,0
Exp/Cntr=0.3,0.1

Type RM Length L Ch R = 1 ,35954   ,424,424,424
BEGIN DESCRIPTION:
Town Creek 64.0
END DESCRIPTION:
XS GIS Cut Line= 4
      1920874.99     13955175.01        1920575.       13955325.
      1920555.99     13955342.43       1919615.7     13955959.55
#Sta/Elev= 30
  4664.6 1922.59  4692.1 1912.52  4711.2 1899.33  4717.9 1879.02  4755.8 1850.32
  4772.6 1840.78  4834.8 1801.34  4872.2 1786.17  4879.9 1784.38    4883 1782.21
  4896.7 1771.79  4901.9 1770.08    4949 1769.45  5000.6 1768.78  5001.1 1768.28
  5016.6 1768.78  5017.5  1770.3  5043.2 1774.09  5123.3 1775.92  5147.3 1777.54
  5154.5 1779.36  5280.1 1779.94  5310.9 1778.49  5600.3 1781.96  5720.7  1784.1
  5825.5 1788.52  5875.7 1788.79  6058.7 1795.44  6117.5  1799.1  6150.5 1800.17
#Mann= 8 ,-1 , 0
  4664.6      .1       0    4883     .07       0    4949    .035       0
  5000.6    .035       0  5016.6    .035       0  5600.3     .07       0
  5720.7    .035       0  6117.5      .1       0
Bank Sta=5000.6,5016.6
XS Rating Curve= 0 ,0
Exp/Cntr=0.3,0.1

Type RM Length L Ch R = 1 ,35530   ,453,453,453
BEGIN DESCRIPTION:
Town Creek 63.0
END DESCRIPTION:
XS GIS Cut Line= 3
      1920724.98       13954975.        1920325.       13955025.
      1919725.03     13955574.98
#Sta/Elev= 30
  4592.3 1898.37  4642.7 1884.04  4696.6 1865.85  4701.7 1860.85  4704.9 1860.77
  4707.8 1856.65  4728.8 1847.37  4731.9  1841.4    4744 1831.92  4750.1 1825.51
  4771.3 1812.06  4792.4 1795.96  4816.6 1789.14  4828.1 1784.34  4834.7 1779.36
  4857.8 1769.11  4959.8 1767.89  4960.3 1767.39  4975.8 1767.89  5033.9 1768.99
  5057.3 1770.59  5173.9 1770.12  5259.4 1776.06  5288.2 1775.05  5434.4  1778.6
  5648.7 1787.92  5713.4 1790.63  5735.5 1791.15  5759.9 1794.09  5809.3 1795.54
#Mann= 7 ,-1 , 0
  4592.3      .1       0  4828.1     .07       0  4959.8     .05       0
  4975.8     .07       0  5033.9    .035       0  5648.7    .063       0
  5713.4    .035       0
Bank Sta=4959.8,4975.8
XS Rating Curve= 0 ,0
Exp/Cntr=0.3,0.1

Type RM Length L Ch R = 1 ,35077   ,400,400,400
BEGIN DESCRIPTION:
Town Creek 62.0
END DESCRIPTION:
XS GIS Cut Line= 3
      1920525.01       13954725.        1919925.       13954875.
      1919324.95       13954825.
#Sta/Elev= 30
  4381.5  1814.1    4388 1812.51  4402.5 1805.37  4417.2 1800.07  4435.7 1795.79
    4479 1788.87    4513 1785.73  4543.9 1780.66  4612.5 1776.35  4642.9 1773.84
  4670.7 1768.67    4680 1765.11  4828.4 1767.31  4896.5 1765.34  4978.8 1765.02
  4979.3 1764.52    4995 1765.02  5076.8 1766.26    5113 1767.66  5120.1 1769.48
  5164.1 1770.95  5233.4 1777.86  5260.5 1777.94  5272.5 1779.69  5323.7 1781.99
  5386.3 1793.33  5453.1 1808.02  5489.3 1817.41  5552.5 1839.82  5602.1 1861.56
#Mann= 6 ,-1 , 0
  4381.5    .035       0  4612.5     .07       0  4978.8     .05       0
    4995     .07       0  5120.1    .035       0  5386.3      .1       0
Bank Sta=4978.8,4995
XS Rating Curve= 0 ,0
Exp/Cntr=0.3,0.1

Type RM Length L Ch R = 1 ,34677   ,341,341,341
BEGIN DESCRIPTION:
Town Creek 61.0
END DESCRIPTION:
XS GIS Cut Line= 3
      1920324.99       13954675.      1919858.43     13954519.31
      1919174.99       13954675.
#Sta/Elev= 30
  4371.1 1779.85  4431.2 1776.52  4722.2 1767.97  4803.9 1766.47  4819.8 1767.45
  4834.1 1770.77  4860.5 1769.76  4865.7 1769.35  4891.7 1768.27  4906.5 1763.74
  4913.2 1761.59  4969.7 1760.46  4970.2 1759.96  4985.9 1760.46  5005.5 1760.77
  5033.2 1770.09  5067.1 1769.62  5079.4 1775.52  5088.6  1777.6  5116.3 1777.78
  5137.8  1781.2  5153.1  1781.4  5177.8 1789.34  5211.7 1791.99  5235.4 1800.02
  5337.8 1832.73  5414.8 1866.04  5451.7 1879.88  5513.2 1909.66  5563.9 1925.82
#Mann= 9 ,-1 , 0
  4371.1    .035       0  4431.2      .1       0  4722.2    .033       0
  4860.5     .07       0  4865.7    .033       0  4906.5     .07       0
  4969.7     .05       0  4985.9     .07       0  5235.4      .1       0
Bank Sta=4969.7,4985.9
XS Rating Curve= 0 ,0
Exp/Cntr=0.3,0.1

Type RM Length L Ch R = 1 ,34336   ,787,787,787
BEGIN DESCRIPTION:
Mapping XS 1ece7bd8
END DESCRIPTION:
XS GIS Cut Line= 3
      1920778.69      13954698.6      1919790.02     13954217.74
      1919199.39     13954256.46
#Sta/Elev= 30
  3784.9 1860.06  3862.1 1843.29  3910.1 1830.19    3945 1828.39  3971.8 1820.36
  4042.1 1813.52  4088.8 1797.09  4135.5 1788.35  4272.3  1778.2  4391.9 1773.84
  4509.1 1770.78  4659.2 1761.89  4705.9 1765.59  4789.4 1765.83  4869.7 1769.17
  4891.9 1764.99  4964.1 1761.49  4985.7 1756.67    4986 1753.88  4986.5 1753.38
  5002.3 1753.88  5036.2 1755.91  5046.3 1763.52  5056.4 1771.65  5177.5 1774.93
  5256.6 1782.31  5345.8 1806.24    5385 1814.45  5466.2 1845.65  5476.2 1853.67
#Mann= 6 ,-1 , 0
  3784.9    .035       0  4391.9     .07       0    4986     .05       0
  5002.3     .07       0  5046.3    .035       0  5256.6      .1       0
Bank Sta=4986,5002.3
XS Rating Curve= 0 ,0
Exp/Cntr=0.3,0.1

Type RM Length L Ch R = 1 ,33549   ,148,148,148
BEGIN DESCRIPTION:
Mapping XS 6671d8f9
END DESCRIPTION:
XS GIS Cut Line= 4
      1920630.17     13953688.64      1920007.12     13953969.11
      1919687.19     13953970.14      1919173.81     13954160.11
#Sta/Elev= 30
  4363.5 1860.15  4442.9 1827.46  4495.4  1813.2  4506.9 1811.81  4527.2 1803.73
  4608.9 1782.75  4683.6 1776.15  4704.3 1769.65  4743.8 1763.89  4849.1 1763.53
  4941.2 1754.21  4957.6 1757.13  4983.9 1756.83  4992.2 1753.37  4992.7 1752.87
  5008.5 1753.37  5187.5 1754.89  5202.5  1760.7  5220.5 1763.83  5421.2 1766.05
  5460.3  1769.2  5533.9 1769.01    5553 1771.56  5671.4 1774.24  5692.3 1777.28
  5732.2 1781.74  5795.9 1802.97    5841 1811.75    5887 1830.61  5914.1  1844.6
#Mann= 7 ,-1 , 0
  4363.5     .07       0  4495.4    .035       0  4683.6     .07       0
  4992.2     .05       0  5008.5     .07       0  5421.2    .035       0
  5692.3      .1       0
Bank Sta=4992.2,5008.5
XS Rating Curve= 0 ,0
Exp/Cntr=0.3,0.1

Type RM Length L Ch R = 1 ,33401   ,114,114,114
BEGIN DESCRIPTION:
Town Creek 60.1
END DESCRIPTION:
XS GIS Cut Line= 6
      1920623.02     13953600.37      1920184.68     13953767.45
      1920097.88     13953813.03      1920071.84     13953823.88
      1919956.82     13953821.71      1919234.13     13954103.84
#Sta/Elev= 30
  4408.9 1875.36  4425.6 1865.06  4454.5  1852.1  4513.3  1832.3  4561.5 1817.14
  4592.4 1808.37  4605.4 1807.76  4682.4 1788.43  4704.9 1786.78  4746.7 1778.56
  4806.5 1776.57  4888.1 1772.54  4973.2 1762.14  5040.3 1758.77  5090.1 1755.74
  5090.6 1755.24  5107.2 1755.74  5152.5 1758.91  5264.7  1760.5  5283.5 1763.44
    5355 1764.52  5462.2 1765.53  5515.9 1766.14  5548.1 1769.48  5618.9 1769.58
    5745 1775.91  5785.4  1779.9  5812.6  1787.3    5854 1802.48  5895.1 1810.57
#Mann= 12 ,-1 , 0
  4408.9      .1       0  4513.3     .07       0  4561.5    .035       0
  4806.5     .07       0  4888.1    .035       0  5040.3     .07       0
  5090.1     .05       0  5107.2     .07       0  5152.5    .035       0
    5355     .07       0  5462.2    .035       0    5745      .1       0
Bank Sta=5090.1,5107.2
XS Rating Curve= 0 ,0
Exp/Cntr=0.3,0.1

Type RM Length L Ch R = 1 ,33287   ,422,422,422
BEGIN DESCRIPTION:
Town Creek 60.0
END DESCRIPTION:
XS GIS Cut Line= 3
      1920624.99     13953425.01        1920025.       13953725.
       1919149.9     13954105.11
#Sta/Elev= 30
  4333.4 1899.84  4429.9 1857.88  4507.3 1831.75  4599.8 1805.79  4652.3 1796.42
  4742.1 1779.41  4866.2 1775.27  4903.1 1763.78  4923.3 1762.22  4976.9 1746.59
  4988.4 1746.42  4989.3 1746.42  4989.8 1745.92  5006.4 1746.42  5013.6 1746.59
    5043 1755.57  5206.9 1760.44  5249.1 1758.98  5291.6 1763.89  5315.9 1764.07
  5424.9 1765.17  5614.7 1769.18  5723.5 1774.04  5775.7  1779.8  5805.1 1788.07
    5828 1798.13  5850.9 1804.86    5900  1814.5  5935.9 1829.22  5958.3 1841.26
#Mann= 10 ,-1 , 0
  4333.4      .1       0  4507.3     .07       0  4652.3    .035       0
  4988.4     .07       0  4989.3     .05       0  5006.4     .07       0
  5206.9    .035       0  5315.9     .07       0  5424.9    .035       0
  5723.5      .1       0
Bank Sta=4989.3,5006.4
XS Rating Curve= 0 ,0
Exp/Cntr=0.3,0.1

Type RM Length L Ch R = 1 ,32865   ,477,477,477
BEGIN DESCRIPTION:
Town Creek 59.0
END DESCRIPTION:
XS GIS Cut Line= 3
      1919975.01       13953325.        1919775.       13953425.
      1919175.03     13954024.97
#Sta/Elev= 30
  4782.5  1774.4  4793.2 1772.11  4807.4  1771.5    4847 1770.24  4927.4 1758.76
  4964.3 1750.28  4965.8 1747.02  4966.3 1746.52  4982.9 1747.02  5001.2  1748.2
  5041.8 1754.67  5138.8 1753.24  5244.9 1757.14  5271.4 1755.79  5285.7 1757.69
  5321.3  1760.2    5352 1761.33  5363.7 1760.19  5390.2 1763.05  5406.6 1762.43
  5470.9 1763.44  5567.3 1765.67  5614.9 1769.36    5666  1771.1  5673.9 1772.64
  5694.6 1774.36  5720.1 1776.08  5758.3 1783.95  5814.5 1803.92  5854.6  1812.7
#Mann= 7 ,-1 , 0
  4782.5    .094       0  4807.4     .07       0  4965.8     .05       0
  4982.9     .07       0  5470.9     .07       0  5614.9    .035       0
  5694.6      .1       0
Bank Sta=4965.8,4982.9
XS Rating Curve= 0 ,0
Exp/Cntr=0.3,0.1

Type RM Length L Ch R = 1 ,32388   ,434,434,434
BEGIN DESCRIPTION:
Town Creek 58.0
END DESCRIPTION:
XS GIS Cut Line= 3
      1919674.97     13952975.02        1919375.       13953225.
      1918924.98     13953825.02
#Sta/Elev= 30
  4609.5 1765.75  4807.6 1763.27  4849.8 1761.37  4881.9 1755.34  4924.7 1746.33
  4938.8 1745.18    4981  1746.3  4996.8 1745.28  4997.4 1744.08  4997.9 1743.58
  5014.6 1744.08    5016 1746.82  5023.9 1748.62    5056 1752.28  5111.8 1752.54
  5168.5  1752.5    5211 1755.16  5254.8 1755.01    5311 1758.65  5340.6  1758.8
  5374.8 1760.15  5445.1 1766.99  5509.3 1773.52  5554.4 1783.07  5601.8 1786.02
  5614.4 1787.45  5640.5 1793.56    5693 1800.57    5723 1809.88    5750 1813.58
#Mann= 8 ,-1 , 0
  4609.5    .035       0  4881.9      .1       0  4997.4     .05       0
  5014.6      .1       0  5111.8     .07       0  5340.6      .1       0
  5445.1     .07       0  5601.8    .035       0
Bank Sta=4997.4,5014.6
XS Rating Curve= 0 ,0
Exp/Cntr=0.3,0.1

Type RM Length L Ch R = 1 ,31954   ,484,484,484
BEGIN DESCRIPTION:
Town Creek 57.0
END DESCRIPTION:
XS GIS Cut Line= 3
      1919474.99       13952925.        1919025.       13952975.
      1918825.01     13953224.99
#Sta/Elev= 30
  4559.4 1761.37  4661.1 1759.02  4710.8  1757.8  4862.8 1757.87  4877.9 1755.71
    4896 1748.57  4914.1 1743.54    4922 1742.24  4943.4 1741.97  4961.5 1742.99
  4971.6 1742.15  4982.6 1743.03  4996.8 1742.13  5006.8  1743.4    5018 1741.83
    5019 1740.81  5019.5 1740.31  5035.7 1740.31  5036.2 1740.81  5037.2 1743.14
  5043.4 1745.88  5058.8  1747.7  5075.6 1747.22  5097.2 1748.44  5104.4 1748.01
  5157.2 1748.76  5176.5 1749.75  5216.3 1752.54  5277.8 1760.23  5332.3 1762.97
#Mann= 4 ,-1 , 0
  4559.4     .07       0  4661.1      .1       0    5019     .05       0
  5036.2      .1       0
Bank Sta=5019,5036.2
XS Rating Curve= 0 ,0
Exp/Cntr=0.3,0.1

Type RM Length L Ch R = 1 ,31470   ,456,456,456
BEGIN DESCRIPTION:
Town Creek 56.0
END DESCRIPTION:
XS GIS Cut Line= 3
      1919475.03       13952725.        1918775.       13952625.
      1918174.96     13952274.98
#Sta/Elev= 30
  4292.4 1762.62  4342.5 1765.45  4348.6 1764.48  4360.7 1759.69  4366.5 1759.17
  4486.4 1754.72  4585.6 1750.32  4696.1 1746.61  4789.2 1747.33  4832.5 1748.44
    4884 1747.76  4937.4 1743.85  4962.8 1743.41  4996.9 1740.38  4997.4 1739.88
  5016.4 1740.38  5092.9 1741.38  5102.8 1746.75  5126.9  1766.3  5137.9 1771.91
  5186.1 1781.56  5228.3 1787.85  5311.7 1797.78  5332.5 1803.11  5367.3 1804.58
  5391.6 1812.58  5429.6 1819.78  5508.6 1842.32  5662.1 1894.35  5694.2  1903.4
#Mann= 7 ,-1 , 0
  4292.4     .07       0  4486.4    .035       0  4585.6     .07       0
  4789.2      .1       0  4937.4     .07       0  4996.9     .05       0
  5016.4     .07       0
Bank Sta=4996.9,5016.4
XS Rating Curve= 0 ,0
Exp/Cntr=0.3,0.1

Type RM Length L Ch R = 1 ,31014   ,449,449,449
BEGIN DESCRIPTION:
Town Creek 55.0
END DESCRIPTION:
XS GIS Cut Line= 4
      1919839.66      13952751.5      1919497.25      13952606.5
        1918925.       13952225.      1918324.97     13952074.99
#Sta/Elev= 30
  3944.7 1771.46  4205.6 1766.11  4434.9 1756.76  4539.9 1749.49  4597.1 1747.55
  4641.2 1744.44    4731 1742.55  4799.5 1743.98  4804.7    1745  4805.6 1743.81
  4874.1 1743.54    4968 1740.71  4968.5 1740.21  4987.5 1740.71  5065.8 1741.57
  5082.8 1751.77  5090.5 1752.92  5100.1  1757.2  5180.2 1760.45  5232.8  1764.4
  5312.9 1775.17  5335.2 1780.11  5393.6 1794.82    5409 1800.41  5436.9 1799.71
  5453.9 1807.07  5498.7 1816.57  5545.4  1829.8  5583.4 1843.23  5622.8 1859.05
#Mann= 7 ,-1 , 0
  3944.7     .07       0  4597.1    .035       0  4641.2     .07       0
    4968     .05       0  4987.5     .07       0  5335.2    .035       0
  5583.4     .07       0
Bank Sta=4968,4987.5
XS Rating Curve= 0 ,0
Exp/Cntr=0.3,0.1

Type RM Length L Ch R = 1 ,30565   ,416,416,416
BEGIN DESCRIPTION:
Town Creek 54.0
END DESCRIPTION:
XS GIS Cut Line= 4
      1920115.28     13952180.76      1919555.38     13952176.42
        1919325.       13952175.      1918725.02     13951825.01
#Sta/Elev= 30
  4209.7 1785.01  4236.6 1778.99  4257.6 1775.81  4266.6 1772.09  4308.6 1771.36
  4330.6 1769.33  4389.8  1767.3  4536.6 1763.93  4554.6 1764.74  4560.6 1763.96
  4704.6 1761.93  4785.6 1762.21  4843.7 1754.58  4899.6 1743.91  4917.6 1743.01
  4929.6 1743.58  4962.1 1740.23  4962.6 1739.73  4981.8 1740.23  5143.8 1741.97
  5165.1 1742.86    5172 1741.52  5207.5 1740.82  5209.7 1741.95  5211.9 1744.43
  5218.4 1748.26  5227.5 1752.27  5532.1 1754.84  5598.1  1756.6  5694.6 1761.96
#Mann= 6 ,-1 , 0
  4209.7    .035       0  4389.8     .07       0  4962.1     .05       0
  4981.8     .07       0  5143.8    .033       0  5227.5     .07       0
Bank Sta=4962.1,4981.8
XS Rating Curve= 0 ,0
Exp/Cntr=0.3,0.1

Type RM Length L Ch R = 1 ,30149   ,466,466,466
BEGIN DESCRIPTION:
Town Creek 53.0
END DESCRIPTION:
XS GIS Cut Line= 3
      1919574.97     13952024.98        1919325.       13951825.
        1918725.       13951775.
#Sta/Elev= 30
  4679.8 1761.47  4711.6 1762.01  4720.1 1761.48  4732.8 1751.61  4736.9 1749.85
  4743.6 1745.04  4747.9 1742.76  4755.3 1742.57  4872.1 1740.81  4941.7 1740.69
  4976.7 1740.32  4977.2 1739.82  4995.9 1739.82  4996.4 1740.32    4997 1741.54
  5004.5 1742.04  5022.6 1745.49  5034.6 1747.08  5041.4 1747.02  5043.7  1747.8
  5055.7  1747.6  5085.8 1748.94  5188.6 1750.98  5310.6 1751.93  5334.7 1752.93
  5337.7 1752.35  5430.7 1754.28  5481.1 1755.55  5541.1 1757.91    5602 1761.93
#Mann= 7 ,-1 , 0
  4679.8     .07       0  4755.3    .033       0  4941.7     .07       0
  4976.7     .05       0  4996.4     .07       0  5430.7    .035       0
  5481.1     .07       0
Bank Sta=4976.7,4996.4
XS Rating Curve= 0 ,0
Exp/Cntr=0.3,0.1
