HEC-RAS study Town Creek.prj: Town Creek Base Level Engineering

--- Town Creek.g01 (geometry) --- (continued)

Type RM Length L Ch R = 1 ,29683   ,834,834,834
BEGIN DESCRIPTION:
Town Creek 52.0
END DESCRIPTION:
XS GIS Cut Line= 3
      1919975.04     13951825.03        1919375.       13951375.
      1918526.37     13951389.43
#Sta/Elev= 30
  4249.6  1762.8  4314.4 1759.92  4426.6 1756.95  4458.6 1757.33  4565.4 1758.27
  4569.1 1757.88    4579 1749.73  4587.9 1742.99  4591.6 1741.97  4666.6 1740.85
  4696.6 1741.76  4796.6 1741.97  4876.7 1740.82  4877.2 1740.32  4896.5 1740.82
  4955.8 1741.15  4981.6 1741.79  4996.6 1740.85  5033.2  1745.2  5088.2 1746.84
  5162.3 1748.04  5180.3 1749.13  5234.3 1749.22  5323.3 1751.97  5527.4 1759.89
  5593.4 1763.29  5644.4 1767.54  5655.7  1767.7  5788.4 1783.09  5848.4 1787.48
#Mann= 8 ,-1 , 0
  4249.6    .035       0  4314.4     .07       0  4458.6      .1       0
    4579    .033       0  4876.7     .05       0  4896.5    .033       0
  4955.8     .07       0  5088.2    .035       0
Bank Sta=4876.7,4896.5
XS Rating Curve= 0 ,0
Exp/Cntr=0.3,0.1

Type RM Length L Ch R = 1 ,28849   ,260,260,260
BEGIN DESCRIPTION:
Town Creek 51.0
END DESCRIPTION:
XS GIS Cut Line= 3
      1920479.42       13950843.        1919675.       13950925.
      1918728.85     13951106.05
#Sta/Elev= 30
  4195.6  1859.8    4266 1842.81  4283.9 1835.16  4296.1 1831.89  4320.2  1819.4
  4338.3 1814.59  4359.5 1803.04  4378.9 1795.59  4395.6 1788.35  4410.7 1785.62
  4443.5 1775.15    4459 1771.58  4480.1 1764.27  4504.2 1761.36  4528.3  1760.4
  4540.4 1758.34  4576.6 1758.96  4630.8 1753.79  4687.9 1753.26  4845.2 1747.52
  4905.3  1746.8  4929.4 1740.72  5246.8 1740.73  5293.8 1740.72  5294.3 1740.22
  5313.6 1740.72  5322.4 1742.75  5347.8 1744.36  5516.8 1747.58  5967.5 1765.12
#Mann= 10 ,-1 , 0
  4195.6     .07       0  4378.9      .1       0  4443.5    .035       0
  4687.9      .1       0  4845.2    .033       0  5246.8     .07       0
  5293.8     .05       0  5313.6     .07       0  5347.8     .07       0
  5516.8    .035       0
Bank Sta=5293.8,5313.6
XS Rating Curve= 0 ,0
Exp/Cntr=0.3,0.1

Type RM Length L Ch R = 1 ,28589   ,193,193,193
BEGIN DESCRIPTION:
Town Creek 51.1
END DESCRIPTION:
XS GIS Cut Line= 4
      1920459.83      13950694.1       1919613.5     13950701.91
      1919454.65     13950707.12      1918720.27      13951066.5
#Sta/Elev= 30
  4114.8 1862.73  4141.2 1851.87  4162.2 1837.45  4174.2 1832.93  4189.2 1823.06
  4207.2 1816.39  4237.2 1800.17  4282.2 1782.27    4309 1774.26  4345.2 1763.28
  4402.2 1757.86  4414.2 1753.59  4450.2 1754.45  4486.2 1749.63  4559.5  1747.4
  4660.9 1745.49  4825.3 1745.44  4861.3 1742.07  4939.3 1739.03  5052.4 1737.78
  5052.9 1737.28  5072.2 1737.78  5098.7 1738.27  5120.1 1739.09    5166 1745.52
  5223.2 1744.02  5326.3 1747.24  5464.9  1747.7    5673 1751.91  5937.7  1764.6
#Mann= 8 ,-1 , 0
  4114.8      .1       0    4309    .035       0  4559.5      .1       0
  4660.9     .07       0  5052.4     .05       0  5072.2     .07       0
  5098.7     .07       0  5464.9    .035       0
Bank Sta=5052.4,5072.2
XS Rating Curve= 0 ,0
Exp/Cntr=0.3,0.1

Type RM Length L Ch R = 1 ,28396   ,568,568,568
BEGIN DESCRIPTION:
Town Creek 50.0
END DESCRIPTION:
XS GIS Cut Line= 3
      1920320.36     13950577.79        1919625.       13950525.
      1918793.03     13950856.39
#Sta/Elev= 30
  4299.5 1785.06  4325.6 1776.18  4358.1 1766.98  4372.7 1760.53  4438.8 1751.08
    4475 1751.66    4502 1748.62  4604.3 1744.59  4776.4 1743.75    4875  1739.1
  4947.3 1731.02  4965.8  1727.1  4992.4 1722.82  5085.5 1722.62    5086 1722.12
  5105.3 1722.62  5179.4 1725.44  5208.5 1735.46  5221.4 1732.25  5234.3  1734.5
  5276.3 1731.13  5300.5 1733.25  5336.9 1731.93  5353.1 1734.13  5366.7 1738.78
  5460.3 1742.81  5724.1 1744.38  5834.7  1748.7  5849.4 1748.25  5892.4 1749.75
#Mann= 10 ,-1 , 0
  4299.5      .1       0  4325.6    .035       0  4776.4     .07       0
    4875    .035       0  4965.8     .07       0  5085.5     .05       0
  5105.3     .07       0  5724.1    .035       0  5834.7     .07       0
  5849.4    .035       0
#XS Ineff= 2 , 0
         4773.63 1744.31
Permanent Ineff=
       F       F
Bank Sta=5085.5,5105.3
XS Rating Curve= 0 ,0
Exp/Cntr=0.3,0.1

Type RM Length L Ch R = 1 ,27828   ,543,543,543
BEGIN DESCRIPTION:
Town Creek 49.0
END DESCRIPTION:
XS GIS Cut Line= 3
        1920425.       13950575.        1919625.       13950025.
      1919191.71     13950004.36
#Sta/Elev= 30
  4024.7  1844.2  4058.2 1823.55  4090.9 1807.21  4102.6 1800.14  4134.6 1786.28
  4157.4 1779.27  4174.7  1773.7  4187.4 1772.34  4229.3 1758.08  4280.3 1753.23
  4287.7 1749.36  4346.2 1749.48  4363.2 1748.57  4400.4 1743.95  4636.6 1737.34
  4709.8 1735.81  4745.1 1728.39  4906.9 1724.87  4935.6 1722.93  4997.1 1721.86
  5009.1 1719.27  5028.8 1719.03  5029.3 1718.53  5049.6 1719.03  5051.2 1727.73
  5063.9 1736.37  5075.2  1744.8  5087.2 1747.06    5130 1746.89  5429.3 1753.16
#Mann= 6 ,-1 , 0
  4024.7      .1       0  4157.4    .035       0  4636.6     .07       0
  5028.8     .05       0  5049.6     .07       0  5063.9    .045       0
Bank Sta=5028.8,5049.6
XS Rating Curve= 0 ,0
Exp/Cntr=0.3,0.1

Type RM Length L Ch R = 1 ,27285   ,562,562,562
BEGIN DESCRIPTION:
Town Creek 48.0
END DESCRIPTION:
XS GIS Cut Line= 3
      1920574.98     13950424.97        1919925.       13949625.
      1919524.95     13949675.01
#Sta/Elev= 30
  3964.6 1891.35  4002.1  1877.5  4079.7 1836.91    4103 1831.43  4122.5 1819.52
  4137.1 1815.46  4174.8 1798.19    4265 1776.57  4320.5 1760.42  4379.4 1748.07
  4407.9 1749.06  4452.8 1744.18  4627.6  1736.2  4690.2 1728.55  4761.6 1726.05
  4812.3 1727.01  4891.7 1723.82  4922.5 1722.21    5006  1715.2  5034.9 1715.06
  5035.4 1714.56  5055.8 1715.06  5072.5 1717.91  5096.7 1717.32  5111.8 1724.84
  5121.7 1733.58    5136 1740.32  5146.5 1741.56  5386.9 1745.58  5398.5 1745.54
#Mann= 10 ,-1 , 0
  3964.6     .07       0    4265    .035       0  4627.6     .07       0
  4761.6    .035       0  4891.7     .07       0  4922.5      .1       0
  5034.9     .05       0  5055.8      .1       0  5146.5     .07       0
  5386.9    .045       0
Bank Sta=5034.9,5055.8
XS Rating Curve= 0 ,0
Exp/Cntr=0.3,0.1

Type RM Length L Ch R = 1 ,26723   ,565,565,565
BEGIN DESCRIPTION:
Town Creek 47.0
END DESCRIPTION:
XS GIS Cut Line= 3
      1920524.99       13949175.        1920125.       13949175.
      1919674.97     13949275.01
#Sta/Elev= 30
  4600.3 1778.34  4645.2 1775.22  4670.9 1772.96    4680 1767.31  4682.9 1766.98
  4727.9 1768.09  4743.8 1765.92  4769.9 1761.43  4805.7 1746.42    4830 1736.47
  4865.9 1727.33  4898.9 1721.67  4913.9 1720.95  4940.9 1715.32  4994.9 1715.04
  4996.5    1712    4997  1711.5  5017.6    1712  5018.3 1713.28  5034.7 1715.69
  5068.5  1713.9  5075.8 1714.73  5092.2 1717.34  5105.4 1725.01  5123.8 1732.26
  5138.9  1734.1  5311.3 1734.29  5421.3  1737.5    5428 1738.93  5461.3 1739.11
#Mann= 9 ,-1 , 0
  4600.3    .035       0  4645.2    .063       0  4743.8    .035       0
  4805.7     .07       0  4996.5     .05       0  5017.6     .07       0
  5075.8    .035       0  5311.3     .07       0  5421.3    .035       0
Bank Sta=4996.5,5017.6
XS Rating Curve= 0 ,0
Exp/Cntr=0.3,0.1

Type RM Length L Ch R = 1 ,26158   ,555,555,555
BEGIN DESCRIPTION:
Town Creek 46.0
END DESCRIPTION:
XS GIS Cut Line= 3
      1920625.05       13948675.        1920225.       13948675.
      1919575.03     13948974.98
#Sta/Elev= 30
    4605  1788.9  4715.6 1782.97  4781.6 1775.88  4802.6 1770.49  4835.6 1770.65
  4862.6 1766.68  4881.8 1759.47  4899.8 1748.79  4911.8 1743.33  4919.3 1736.89
  4937.6 1725.77  4950.8 1716.02  4964.6 1712.34  4966.1 1707.28  4966.6 1706.78
  4987.2 1707.28  4997.6 1708.04  5000.6 1711.19  5004.5 1712.82  5016.7 1714.05
  5069.6 1712.57  5115.8 1714.95  5129.1  1717.4  5148.9 1726.35  5168.7 1729.79
  5579.1  1732.7  5618.1 1733.47  5660.9 1738.85  5697.4 1741.78  5720.9  1741.2
#Mann= 6 ,-1 , 0
    4605    .035       0  4919.3     .07       0  4966.1     .05       0
  4987.2     .07       0  5004.5    .035       0  5579.1     .07       0
Bank Sta=4966.1,4987.2
XS Rating Curve= 0 ,0
Exp/Cntr=0.3,0.1

Type RM Length L Ch R = 1 ,25603   ,427,427,427
BEGIN DESCRIPTION:
Town Creek 45.0
END DESCRIPTION:
XS GIS Cut Line= 3
      1920525.02     13948375.01        1920125.       13948175.
      1919324.99       13948125.
#Sta/Elev= 30
  4560.9  1778.5  4571.2 1777.49  4605.5 1774.99  4614.4  1772.8  4623.1 1767.77
  4672.5 1769.98  4690.7 1766.98  4710.3 1765.71  4724.5 1762.54  4763.9 1759.04
  4797.5 1753.95  4827.7 1751.94  4847.8 1745.74  4907.7  1716.5  4938.4 1711.46
  4963.2  1709.4  4964.7 1706.55  4965.2 1706.05  4985.8 1706.55  5015.4 1707.28
  5047.8 1707.79  5098.9  1716.5    5147 1720.94  5180.1 1725.74  5234.2 1723.33
  5474.7  1727.4    5607 1731.39  5705.6 1737.95  5796.3 1744.02  5809.7 1746.78
#Mann= 9 ,-1 , 0
  4560.9    .035       0  4571.2    .063       0  4690.7      .1       0
  4907.7     .07       0  4964.7     .05       0  4985.8     .07       0
  5015.4    .035       0    5607     .07       0  5705.6    .035       0
Bank Sta=4964.7,4985.8
XS Rating Curve= 0 ,0
Exp/Cntr=0.3,0.1

Type RM Length L Ch R = 1 ,25176   ,110,110,110
BEGIN DESCRIPTION:
Town Creek 44.1
END DESCRIPTION:
XS GIS Cut Line= 5
       1920970.3     13947647.22      1920165.59     13947780.04
      1920032.77      13947816.5      1919936.42     13947842.54
      1919163.02     13947858.16
#Sta/Elev= 30
  4041.2 1786.08  4165.7 1779.96  4189.5 1778.94  4278.3 1768.99    4290  1769.1
  4311.7 1768.82  4390.4 1760.85  4498.4 1737.31  4536.7 1741.94    4561 1739.02
  4679.6  1734.2  4769.7 1726.28  4893.7 1713.49  4996.8  1707.6    5007  1707.5
  5007.5    1707  5028.3  1707.5  5104.2 1712.57  5125.4 1711.48  5146.4 1714.82
  5228.3 1720.55  5239.5 1720.72  5470.4 1726.24  5634.5 1736.07  5698.4 1742.52
  5722.1 1746.57  5758.5 1756.23  5810.9 1763.68  5853.4 1770.03  5867.9 1771.42
#Mann= 15 ,-1 , 0
  4041.2     .07       0  4165.7    .035       0  4189.5    .063       0
    4290    .035       0  4390.4     .07       0  4769.7    .035       0
  4893.7     .07       0  4996.8     .07       0    5007     .05       0
  5028.3     .07       0  5228.3     .07       0  5239.5    .035       0
  5634.5     .07       0  5810.9    .035       0  5853.4     .07       0
Bank Sta=5007,5028.3
XS Rating Curve= 0 ,0
Exp/Cntr=0.3,0.1

Type RM Length L Ch R = 1 ,25066   ,547,547,547
BEGIN DESCRIPTION:
Town Creek 44.0
END DESCRIPTION:
XS GIS Cut Line= 3
      1920575.03     13947574.99        1919975.       13947725.
      1919174.95       13947775.
#Sta/Elev= 30
  4386.1 1762.99  4411.5 1760.76  4443.5  1752.4  4482.6 1749.29  4510.4 1741.59
  4550.6 1738.93  4584.6 1733.81    4597 1735.46  4674.3 1731.03  4769.2 1728.42
  4841.4 1722.46  4859.9 1719.84  4884.4 1712.34  4912.4 1708.11  4943.8 1707.09
  4963.7 1703.77  4997.5  1703.3    4998  1702.8  5018.8  1703.3  5020.2 1708.12
  5056.3 1711.71  5238.3  1717.3  5332.8  1720.8  5383.9 1724.89  5453.1 1726.25
  5534.2 1733.36  5603.8 1736.43  5729.6 1760.07  5768.7 1764.27  5806.2 1770.68
#Mann= 7 ,-1 , 0
  4386.1     .07       0  4841.4    .035       0  4943.8     .07       0
  4997.5     .05       0  5018.8     .07       0  5238.3    .035       0
  5603.8     .07       0
Bank Sta=4997.5,5018.8
XS Rating Curve= 0 ,0
Exp/Cntr=0.3,0.1

Type RM Length L Ch R = 1 ,24519   ,572,572,572
BEGIN DESCRIPTION:
Town Creek 43.0
END DESCRIPTION:
XS GIS Cut Line= 3
      1920624.96     13947524.99        1919825.       13947225.
      1919024.98     13947575.01
#Sta/Elev= 30
  4145.2 1768.27    4212 1762.89  4304.9 1744.33  4330.6  1742.9  4372.2  1729.9
    4526 1724.39  4536.4 1721.74  4658.6  1720.3  4762.7 1719.27  4881.3  1718.6
  4926.5 1704.25  4963.9 1700.46  4964.4 1699.96  4985.2 1700.46  4988.4 1700.55
    5064 1703.88  5147.7 1708.84  5304.7  1713.4  5383.3 1727.15  5495.6 1734.71
    5570 1739.21  5602.7  1747.3    5642 1750.56  5671.9  1757.9  5724.4 1764.27
  5746.8 1766.73  5766.5 1773.02  5802.5  1768.1  5819.9 1774.18  5872.8 1780.87
#Mann= 11 ,-1 , 0
  4145.2    .035       0  4658.6     .07       0  4762.7      .1       0
  4963.9     .05       0  4985.2      .1       0  4988.4     .07       0
    5064      .1       0  5147.7     .07       0  5495.6    .035       0
  5724.4     .07       0  5819.9    .035       0
Bank Sta=4963.9,4985.2
XS Rating Curve= 0 ,0
Exp/Cntr=0.3,0.1

Type RM Length L Ch R = 1 ,23947   ,764,764,764
BEGIN DESCRIPTION:
Town Creek 42.0
END DESCRIPTION:
XS GIS Cut Line= 3
        1920575.       13947425.        1919775.       13946725.
        1918975.       13945975.
#Sta/Elev= 30
  3941.6 1763.86  4011.6 1754.16    4018 1751.45  4022.2 1744.72  4038.1 1745.47
  4064.7 1744.27  4086.1  1735.6  4119.4  1728.8    4193  1719.3  4246.8 1717.16
    4348  1712.7  4573.6 1707.34  4723.7 1709.96  4860.7  1707.5  4890.4 1704.94
  4983.9 1697.76  4984.4 1697.26  5005.7 1697.76  5038.4 1701.38  5067.7 1722.14
  5089.4 1727.13  5299.7 1733.22  5364.3 1735.44  5488.7 1739.73    5656 1757.36
    5747 1778.32  5936.1  1850.2  6033.4 1892.84  6073.2    1905  6101.2 1908.25
#Mann= 15 ,-1 , 0
  3941.6    .035       0  4038.1      .1       0  4119.4     .07       0
    4193      .1       0  4246.8     .07       0    4348      .1       0
  4860.7     .07       0  4890.4      .1       0  4983.9     .05       0
  5005.7      .1       0  5089.4     .07       0  5299.7    .035       0
  5364.3     .07       0  5488.7      .1       0  6073.2     .07       0
#XS Ineff= 2 , 0
            4723  1710.3
Permanent Ineff=
       F       F
Bank Sta=4983.9,5005.7
XS Rating Curve= 0 ,0
Exp/Cntr=0.3,0.1

Type RM Length L Ch R = 1 ,23183   ,364,364,364
BEGIN DESCRIPTION:
Town Creek 41.0
END DESCRIPTION:
XS GIS Cut Line= 5
      1920605.03     13947403.43      1920421.02     13946832.29
      1920466.16     13946729.86      1920394.98     13946330.55
      1919710.97     13945738.56
#Sta/Elev= 30
  4337.4 1766.15  4378.5 1763.97  4441.7    1759  4492.3 1752.51  4625.9 1719.95
  4653.8 1715.65  4708.9  1712.2  4749.2 1706.15  4790.1 1704.57  4811.2 1703.83
  4859.1 1700.11  4941.2 1700.28  4970.7 1693.42  4999.1 1692.28  4999.6 1691.78
    5021 1692.28  5032.1 1693.37  5067.7 1698.49  5080.6 1706.58    5089  1712.9
  5098.2 1717.01  5216.1 1716.18  5303.7 1715.63  5382.5 1715.01    5764 1715.42
  5878.4 1717.19  5959.2 1722.67  6262.3 1731.76  6292.9 1733.29  6359.6  1740.8
#Mann= 14 ,-1 , 0
  4337.4    .035       0  4378.5      .1       0  4708.9     .07       0
  4790.1      .1       0  4811.2     .07       0  4999.1     .05       0
    5021     .07       0  5032.1    .035       0  5080.6      .1       0
  5216.1    .035       0  5303.7      .1       0  5382.5    .035       0
    5764     .07       0  6262.3      .1       0
#XS Ineff= 2 , 0
                         5108.89         1717.62
Permanent Ineff=
       F       F
Bank Sta=4999.1,5021
XS Rating Curve= 0 ,0
Exp/Cntr=0.3,0.1

Type RM Length L Ch R = 1 ,22819   ,579,579,579
BEGIN DESCRIPTION:
Town Creek 40.0
END DESCRIPTION:
XS GIS Cut Line= 3
      1920974.98     13947124.96        1920775.       13946775.
      1920524.99     13946424.99
#Sta/Elev= 30
  4597.2 1770.13  4663.9 1765.37  4710.2 1761.08  4730.9 1756.68  4763.6 1748.09
  4795.6 1740.14  4852.1 1730.77  4865.7 1728.15  4874.8 1725.12  4894.5 1716.25
  4923.1 1698.61  4934.8  1694.2  4951.7 1690.72  4964.9 1689.55  4965.4 1689.05
  4986.8 1689.55  4986.9 1692.44  5000.5 1693.62  5034.8 1690.84  5037.3 1690.85
  5060.3    1697    5084 1699.87  5103.7 1703.87  5111.1 1704.53  5182.9 1707.84
  5206.9 1710.25  5232.3 1711.22  5292.6 1715.61  5375.7 1715.37  5430.4 1715.18
#Mann= 8 ,-1 , 0
  4597.2    .035       0  4663.9      .1       0  4763.6     .07       0
  4852.1      .1       0  4964.9     .05       0  4986.8      .1       0
  5034.8    .035       0  5375.7      .1       0
Bank Sta=4964.9,4986.8
XS Rating Curve= 0 ,0
Exp/Cntr=0.3,0.1

Type RM Length L Ch R = 1 ,22240   ,588,588,588
BEGIN DESCRIPTION:
Town Creek 39.0
END DESCRIPTION:
XS GIS Cut Line= 3
      1921274.98     13946724.97        1921075.       13946375.
      1920625.05     13946325.01
#Sta/Elev= 30
  4597.1 1744.18  4647.4 1741.48  4744.5 1736.82  4774.6 1734.85  4792.6 1731.11
  4802.3    1724  4809.2 1717.45  4819.5 1713.22  4835.6  1704.3  4856.3  1697.1
  4865.1 1691.99  4873.9 1689.22  4908.7 1687.82  4931.1 1688.77  4957.2 1686.85
  4957.7 1686.35  4979.1 1686.85  5020.9 1688.54    5033 1690.69  5060.1 1691.56
  5081.3 1695.16  5120.5 1698.14  5195.5 1698.96    5208  1697.7  5253.3 1698.76
  5277.5 1697.93  5334.8 1703.03  5374.1 1709.59  5401.2 1711.84  5452.9 1713.82
#Mann= 7 ,-1 , 0
  4597.1    .035       0  4647.4     .07       0  4744.5      .1       0
  4835.6     .07       0  4957.2     .05       0  4979.1     .07       0
  5195.5    .035       0
Bank Sta=4957.2,4979.1
XS Rating Curve= 0 ,0
Exp/Cntr=0.3,0.1

Type RM Length L Ch R = 1 ,21652   ,564,564,564
BEGIN DESCRIPTION:
Town Creek 38.0
END DESCRIPTION:
XS GIS Cut Line= 3
      1921074.98     13945725.01        1920725.       13945925.
        1920525.       13946275.
#Sta/Elev= 30
  4600.8 1708.59  4640.4 1708.39  4653.9 1707.81  4704.9 1706.55  4745.4 1696.07
  4762.7 1696.97  4783.4 1696.66  4804.8 1694.24  4842.2 1692.44  4890.5  1687.9
  4918.2 1687.27  4938.9 1685.79  4952.7  1686.3  4966.6 1684.62    4972  1682.8
  4972.5  1682.3  4993.4  1682.3  4993.9  1682.8  4994.2 1684.42  5001.1 1686.14
  5004.9 1688.45  5007.1 1690.98  5011.1 1694.15  5018.7 1698.85  5023.2 1700.08
  5042.3 1707.27  5063.6 1710.86  5234.9 1712.87  5370.2 1713.76    5407 1713.88
#Mann= 5 ,-1 , 0
  4600.8     .07       0  4653.9     .07       0    4972     .05       0
  4993.9     .07       0  5370.2      .1       0
Bank Sta=4972,4993.9
XS Rating Curve= 0 ,0
Exp/Cntr=0.3,0.1

Type RM Length L Ch R = 1 ,21088   ,572,572,572
BEGIN DESCRIPTION:
Town Creek 37.0
END DESCRIPTION:
XS GIS Cut Line= 3
        1921125.       13945575.        1920775.       13945375.
      1920375.03       13945425.
#Sta/Elev= 30
  4596.8 1708.27  4671.2 1707.46  4724.1 1706.11  4743.8  1705.8  4760.8 1703.51
  4771.8 1700.69  4805.9 1690.29  4864.7 1689.27  4875.1  1690.3  4897.1 1688.93
  4913.1 1689.29  4938.9 1687.31  4941.8 1686.47  4969.7 1683.02  4971.2 1680.42
  4971.7 1679.92  4992.7 1679.92  4993.2 1680.42  5014.6 1681.21  5020.7 1683.38
  5024.8  1685.5  5026.7 1686.31  5035.8 1693.64  5041.8 1702.16  5044.9 1704.12
    5063 1707.98  5090.2 1707.32  5221.6 1708.26  5280.7 1707.58    5403 1709.38
#Mann= 6 ,-1 , 0
  4596.8     .07       0  4724.1     .07       0  4971.2     .05       0
  4993.2     .07       0  5024.8    .035       0  5221.6     .07       0
Bank Sta=4971.2,4993.2
XS Rating Curve= 0 ,0
Exp/Cntr=0.3,0.1

Type RM Length L Ch R = 1 ,20516   ,690,690,690
BEGIN DESCRIPTION:
Town Creek 36.0
END DESCRIPTION:
XS GIS Cut Line= 3
      1921274.98     13945174.98        1920975.       13944875.
      1920574.95     13944925.01
#Sta/Elev= 30
  4575.7 1712.01    4616 1713.53  4654.1  1707.5  4684.9 1706.24  4788.9 1704.96
  4917.2 1705.45  4928.9 1701.83    4948 1692.29  4977.7 1683.73  4981.9  1680.1
  4987.3  1678.8  4987.8 1677.48  4988.3 1676.98  5009.9 1677.48  5013.5 1678.84
    5068 1679.39  5113.3  1682.9  5125.4 1681.64  5130.2    1680  5140.5 1680.63
  5146.6 1684.38  5152.6 1686.25  5161.7 1688.23  5179.8 1689.13  5202.8 1697.27
  5219.4 1700.58  5228.2 1701.39  5250.5 1700.38  5291.5 1703.19  5403.1 1705.89
#Mann= 4 ,-1 , 0
  4575.7     .07       0  4987.8     .05       0  5009.9     .07       0
  5219.4     .07       0
Bank Sta=4987.8,5009.9
XS Rating Curve= 0 ,0
Exp/Cntr=0.3,0.1

Type RM Length L Ch R = 1 ,19826   ,616,616,616
BEGIN DESCRIPTION:
Town Creek 35.0
END DESCRIPTION:
XS GIS Cut Line= 3
      1921236.73     13944406.39       1921000.7     13944267.37
        1920625.       13944125.
#Sta/Elev= 30
  4699.1 1701.52  4896.7 1699.94  4922.6  1701.7    4935 1699.12  4941.9 1691.95
  4956.7 1687.35  4966.3 1678.69  4982.8 1675.43  4983.3 1674.93  5005.1 1675.43
  5030.1 1685.25  5032.4 1689.78  5034.2 1690.88  5037.4 1690.23  5044.8 1692.43
  5059.9 1693.81  5113.9 1692.97  5120.8 1691.51  5132.5 1683.86  5140.1 1683.15
  5153.4 1685.11  5167.4 1684.77  5217.1 1701.59  5253.1  1701.1    5278  1700.9
  5307.2 1695.71  5318.6 1695.33    5341 1702.64  5357.3 1704.27  5374.8 1704.98
#Mann= 6 ,-1 , 0
  4699.1     .07       0  4982.8     .05       0  5005.1     .07       0
  5044.8    .063       0  5253.1    .035       0  5357.3     .07       0
#XS Ineff= 2 , 0
                         5060.34         1693.75
Permanent Ineff=
       F       F
Bank Sta=4982.8,5005.1
XS Rating Curve= 0 ,0
Exp/Cntr=0.3,0.1

Type RM Length L Ch R = 1 ,19210   ,329,329,329
BEGIN DESCRIPTION:
Town Creek 34.0
END DESCRIPTION:
XS GIS Cut Line= 3
      1921675.02       13943725.      1920985.26     13943702.88
      1920574.97       13943725.
#Sta/Elev= 30
  4299.6  1729.4  4334.3 1726.11  4401.2 1719.93  4491.2 1708.24  4542.2 1707.46
  4557.2 1704.17  4641.3 1695.84  4722.8 1690.88  4833.4 1687.04  4893.9 1681.85
  4932.4 1680.47  4944.4 1679.51  4953.4 1677.14  4959.4 1677.97  4971.5 1676.55
  4987.4  1673.9  4988.4 1670.31  4988.9 1669.81  5017.8 1670.31  5025.5  1674.4
  5037.5 1675.88  5052.6 1674.95  5070.6 1676.07  5114.8 1684.34  5157.7 1696.77
  5169.7 1699.07  5262.9  1702.6  5304.9 1716.08    5332 1721.54  5400.6 1720.46
#Mann= 6 ,-1 , 0
  4299.6     .07       0  4334.3    .035       0  4893.9      .1       0
  4988.4     .05       0  5017.8      .1       0  5114.8    .035       0
Bank Sta=4988.4,5017.8
XS Rating Curve= 0 ,0
Exp/Cntr=0.3,0.1

Type RM Length L Ch R = 1 ,18881   ,215,215,215
BEGIN DESCRIPTION:
Town Creek 33.0
END DESCRIPTION:
XS GIS Cut Line= 3
      1921574.97       13943375.        1920975.       13943375.
      1920575.06     13943674.96
#Sta/Elev= 30
  4404.6 1728.02  4426.7 1726.16  4457.1 1722.87  4493.1 1714.52  4604.2 1695.79
  4613.1 1695.71  4676.1 1688.46  4722.5 1686.89  4751.1 1686.67  4831.8 1681.95
    4889 1678.23  4916.1 1673.75  4961.1 1674.53  4964.1 1674.21  4970.4 1670.37
  4970.9 1669.87  4999.8 1670.37  5000.1 1671.84  5010.2 1672.65  5032.7 1672.26
  5055.2 1674.39  5085.2 1685.17  5100.2 1685.55  5118.9 1694.03  5129.5 1696.54
  5212.7  1699.3  5396.4 1701.28  5454.5 1719.72  5474.5 1722.77  5504.5 1722.33
#Mann= 7 ,-1 , 0
  4404.6     .07       0  4426.7      .1       0  4604.2     .07       0
  4722.5    .035       0  4831.8      .1       0  4970.4     .05       0
  4999.8      .1       0
Bank Sta=4970.4,4999.8
XS Rating Curve= 0 ,0
Exp/Cntr=0.3,0.1

Type RM Length L Ch R = 1 ,18666   ,366,366,366
BEGIN DESCRIPTION:
Town Creek 32.1
END DESCRIPTION:
XS GIS Cut Line= 2
      1921730.16     13942569.15      1920674.92     13943476.05
#Sta/Elev= 30
  4070.2 1723.39  4132.8 1721.99  4158.1 1722.49  4183.5 1725.75  4217.4 1725.05
  4252.5 1721.92  4276.7 1718.07  4336.1 1712.53  4464.2 1705.25  4553.6 1702.66
  4593.2 1699.65  4616.1  1694.2  4625.3 1689.65  4656.5 1680.71  4712.8 1678.23
  4786.4 1677.76  4848.4  1676.4  4873.9 1674.57  4933.4 1674.06  4989.8 1669.72
  4990.3 1669.22  5019.3 1669.72  5020.4 1672.13  5030.4 1673.03  5079.8 1674.05
  5099.5 1677.64  5139.1 1690.26  5154.9 1694.34  5166.8 1696.14  5461.6 1699.88
#Mann= 3 ,-1 , 0
  4070.2      .1       0  4989.8     .05       0  5019.3      .1       0
Bank Sta=4989.8,5019.3
XS Rating Curve= 0 ,0
Exp/Cntr=0.3,0.1

Type RM Length L Ch R = 1 ,18300   ,565,565,565
BEGIN DESCRIPTION:
Town Creek 32.0
END DESCRIPTION:
XS GIS Cut Line= 3
      1921794.66     13942142.92        1921075.       13942825.
      1920725.04     13943024.98
#Sta/Elev= 30
  4008.5 1725.82  4067.2 1723.59    4311 1715.22  4421.4 1711.88  4460.7 1709.45
    4490 1709.46  4576.3 1705.26  4628.4 1703.09  4716.4  1699.2  4747.8 1696.72
  4766.7 1691.52  4813.3 1676.89  4825.7 1675.28  4856.4 1674.29  4908.4 1671.61
  4945.6  1672.4  4953.9 1671.17  4955.9 1667.88  4956.4 1667.38    4986 1667.88
  5006.4 1668.66  5016.7 1671.14  5030.5 1672.59  5048.7 1672.64    5072 1678.31
  5085.8 1680.24  5113.5 1688.48  5127.3 1690.42  5158.4 1691.73  5403.1 1695.08
#Mann= 11 ,-1 , 0
  4008.5     .07       0  4067.2    .063       0    4311     .07       0
    4490    .063       0  4576.3     .07       0  4628.4    .063       0
  4716.4    .035       0  4766.7    .094       0  4856.4      .1       0
  4955.9     .05       0    4986      .1       0
Bank Sta=4955.9,4986
XS Rating Curve= 0 ,0
Exp/Cntr=0.3,0.1

Type RM Length L Ch R = 1 ,17735   ,507,507,507
BEGIN DESCRIPTION:
Town Creek 31.0
END DESCRIPTION:
XS GIS Cut Line= 3
      1921425.01       13942325.        1921025.       13942275.
       1920310.2     13942881.26
#Sta/Elev= 30
  4602.3 1706.06  4727.8 1701.21  4863.2 1693.43  4878.9 1691.04  4893.9 1683.46
  4903.1 1680.32  4909.2 1676.96  4924.3 1673.17  4939.6 1671.06  4971.8 1668.82
  5002.8 1664.35  5003.3 1663.85  5032.9 1664.35  5033.6 1668.97  5087.3 1671.29
  5132.7 1675.29    5143 1677.04  5150.5 1677.12  5179.1 1677.94    5220 1676.87
  5293.2 1681.23  5333.1 1682.32  5409.4 1688.34  5458.4 1688.09  5537.1 1691.01
  5757.9 1693.99  5820.4  1697.1  5868.5 1697.64  5910.8 1697.46  5942.7 1698.42
#Mann= 7 ,-1 , 0
  4602.3     .07       0  4863.2      .1       0  5002.8     .05       0
  5032.9      .1       0  5150.5    .035       0  5757.9     .12       0
  5868.5    .063       0
Bank Sta=5002.8,5032.9
XS Rating Curve= 0 ,0
Exp/Cntr=0.3,0.1

Type RM Length L Ch R = 1 ,17228   ,529,529,529
BEGIN DESCRIPTION:
Town Creek 30.0
END DESCRIPTION:
XS GIS Cut Line= 3
      1921595.19     13941802.07        1920775.       13941875.
      1919979.17     13942498.15
#Sta/Elev= 30
  4172.2 1705.59  4351.9 1698.42  4549.8 1691.07  4786.5 1689.38  4992.1 1690.86
  4995.6 1689.86  4998.8 1685.91  5001.7 1678.55  5002.6  1675.3  5002.7 1663.52
  5003.2 1663.02  5032.9 1663.52  5068.6 1667.59    5088 1667.43  5106.4 1664.95
    5117 1665.19  5121.4 1666.69  5143.6  1670.5    5200 1670.83  5204.8 1672.11
  5238.8 1672.54  5326.5  1676.7  5520.8 1689.99  5788.7 1697.95  5821.8 1697.72
  5833.2 1694.88  5913.3 1698.29  5931.2 1696.46  5947.5 1702.85  6006.4 1705.95
#Mann= 6 ,-1 , 0
  4172.2     .07       0  4351.9    .035       0  4786.5     .07       0
  5002.7     .05       0  5032.9     .07       0  5121.4    .035       0
#XS Ineff= 2 , 0
         4986.51 1691.84
Permanent Ineff=
       F       F
Bank Sta=5002.7,5032.9
XS Rating Curve= 0 ,0
Exp/Cntr=0.3,0.1

Type RM Length L Ch R = 1 ,16699   ,551,551,551
BEGIN DESCRIPTION:
Town Creek 29.0
END DESCRIPTION:
XS GIS Cut Line= 3
      1921394.46     13941338.47        1920375.       13941575.
      1919344.49     13941815.29
#Sta/Elev= 30
  3964.7 1694.87  4267.8 1695.68    4366 1687.39  4549.3 1686.62  4721.8 1688.08
  4846.5 1687.49  4904.9 1682.84  4917.6 1677.02  4932.7 1664.95  4979.1 1662.29
  4979.6 1661.79  5009.5 1662.29  5062.1 1662.83  5102.1 1667.41  5117.5  1666.7
  5154.5 1676.11  5194.5 1678.96  5219.1 1688.59  5345.5 1687.38  5467.2 1690.04
  5671.2 1693.79  5685.4 1693.83  5739.8 1694.09    5786 1701.57  5859.9 1707.93
  5915.4 1720.98  5930.8 1721.79  5955.4 1729.51    6017 1743.18  6069.4 1748.93
#Mann= 10 ,-1 , 0
  3964.7     .07       0  4549.3    .035       0  4721.8     .07       0
  4917.6    .035       0  4979.1    .035       0  5009.5    .035       0
  5219.1    .094       0  5467.2     .12       0  5671.2      .1       0
  5685.4     .07       0
Bank Sta=4979.1,5009.5
XS Rating Curve= 0 ,0
Exp/Cntr=0.3,0.1

Type RM Length L Ch R = 1 ,16148   ,569,569,569
BEGIN DESCRIPTION:
Town Creek 28.0
END DESCRIPTION:
XS GIS Cut Line= 3
      1920624.97       13941075.        1920175.       13941125.
        1919375.       13941075.
#Sta/Elev= 30
  4542.5 1692.74  4568.2 1691.83  4604.6 1685.41  4633.4 1680.62  4686.8  1678.8
  4709.5 1674.07    4726 1675.28  4825.6  1672.8  4931.3 1668.18  4979.6  1663.9
  4997.5 1659.97    4998 1659.47    5028 1659.97  5069.9 1662.53  5090.9 1684.83
    5130 1686.52    5157 1681.38  5221.6 1685.07  5232.2 1684.23  5250.2  1688.5
  5373.5 1694.83  5418.7 1699.42  5521.6 1713.77  5549.3 1725.03  5566.3 1728.15
    5623 1731.89    5638 1737.03  5676.6  1755.2  5761.2 1778.69  5796.8 1792.01
#Mann= 9 ,-1 , 0
  4542.5     .07       0  4604.6    .035       0    4726     .07       0
  4825.6    .035       0  4997.5    .035       0    5028    .035       0
  5221.6     .07       0  5418.7      .1       0  5521.6     .07       0
Bank Sta=4997.5,5028
XS Rating Curve= 0 ,0
Exp/Cntr=0.3,0.1

Type RM Length L Ch R = 1 ,15579   ,464,464,464
BEGIN DESCRIPTION:
Town Creek 27.0
END DESCRIPTION:
XS GIS Cut Line= 3
      1920675.02     13940875.01        1920275.       13940625.
      1919925.02     13939925.04
#Sta/Elev= 30
  4521.9 1693.86  4574.3 1691.66  4624.6 1683.24  4668.2 1678.68  4675.8 1676.28
  4715.2 1675.45  4739.5 1672.66  4782.5  1671.8  4959.9 1666.96  4993.6 1660.44
  5009.6 1659.93  5010.1 1659.43  5040.3 1659.93  5057.9 1660.92  5086.4 1661.26
  5105.5 1669.16  5118.9 1677.38  5128.9 1680.13  5164.7 1683.38  5292.1  1688.1
  5360.4 1696.83  5447.1 1713.91  5513.5 1733.73  5554.9 1753.53  5601.9 1768.15
  5621.8 1771.14  5695.8 1782.66    5736 1796.55  5757.2 1801.55  5776.2 1803.06
#Mann= 9 ,-1 , 0
  4521.9     .07       0  4574.3    .035       0  4715.2     .07       0
  4782.5      .1       0  5009.6     .05       0  5040.3      .1       0
  5057.9    .035       0  5447.1      .1       0  5621.8    .035       0
Bank Sta=5009.6,5040.3
XS Rating Curve= 0 ,0
Exp/Cntr=0.3,0.1

Type RM Length L Ch R = 1 ,15115   ,624,624,624
BEGIN DESCRIPTION:
Town Creek 26.0
END DESCRIPTION:
XS GIS Cut Line= 3
      1921125.01     13940575.01      1920517.57     13940245.64
      1920175.01     13939925.01
#Sta/Elev= 30
  4336.8 1694.45  4483.2 1685.11    4575 1683.21  4640.3 1680.79  4750.5 1680.02
    4832 1681.29  4840.2 1679.69  4879.3 1679.83  4889.1 1677.16  4912.5 1668.37
  4956.8 1665.23  4978.4 1659.95  4978.9 1659.45  5009.1 1659.95  5020.2  1660.2
  5110.1 1661.28  5123.1 1663.15  5174.1 1671.28  5195.3 1681.44  5222.5 1687.58
  5237.7  1689.5  5292.9 1690.54  5326.9 1711.61  5344.3 1719.95  5353.6 1721.23
  5365.1 1722.45  5421.1 1749.72  5469.1  1767.3  5484.7 1770.15    5497 1771.68
#Mann= 13 ,-1 , 0
  4336.8     .07       0    4575      .1       0  4640.3     .07       0
  4750.5    .035       0  4889.1     .07       0  4978.4     .05       0
  5009.1     .07       0  5020.2      .1       0  5123.1    .035       0
  5222.5    .063       0  5353.6    .035       0  5421.1      .1       0
  5484.7    .035       0
Bank Sta=4978.4,5009.1
XS Rating Curve= 0 ,0
Exp/Cntr=0.3,0.1

Type RM Length L Ch R = 1 ,14491   ,540,540,540
BEGIN DESCRIPTION:
Town Creek 25.0
END DESCRIPTION:
XS GIS Cut Line= 3
      1921315.58     13940450.25        1920775.       13939775.
      1920325.02     13939575.01
#Sta/Elev= 30
  4134.8 1693.69  4184.1 1690.49  4269.5 1678.94  4658.9 1677.71  4757.7 1677.63
    4815 1673.96    4855 1674.32  4880.7 1661.95  4893.4 1658.43  4988.6 1653.91
  4989.1 1653.41  5019.4 1653.91  5022.1 1656.13    5055 1660.04  5100.2 1675.15
  5115.3 1680.71  5133.5 1690.59  5147.1 1693.63    5206 1689.94  5213.1 1691.04
  5248.7 1712.62  5262.4 1717.24  5283.5 1722.23  5302.7 1730.02  5319.9 1735.46
  5366.9 1742.67  5399.4 1752.22  5433.5 1757.24  5465.4 1768.84  5492.2 1771.07
#Mann= 8 ,-1 , 0
  4134.8      .1       0  4658.9    .035       0    4815      .1       0
  4988.6     .05       0  5019.4      .1       0  5100.2    .063       0
  5262.4    .094       0  5302.7      .1       0
Bank Sta=4988.6,5019.4
XS Rating Curve= 0 ,0
Exp/Cntr=0.3,0.1

Type RM Length L Ch R = 1 ,13951   ,585,585,585
BEGIN DESCRIPTION:
Town Creek 24.0
END DESCRIPTION:
XS GIS Cut Line= 3
      1921824.98     13940174.98        1921125.       13939375.
        1920575.       13939275.
#Sta/Elev= 30
    3937 1687.43  4004.1 1684.25  4085.1 1678.68  4473.9 1675.98  4619.2 1674.58
  4676.2 1673.53  4732.5 1672.49  4803.4 1668.57  4828.1    1665  4841.8 1665.66
  4870.1 1664.19    4899 1656.45  4982.3 1653.09  4982.8 1652.59  5013.1 1653.09
  5080.8 1658.85  5108.2 1665.99  5123.5 1666.41  5135.9 1669.69  5155.2 1674.27
  5235.5 1680.95  5254.6 1682.55  5263.7 1679.21  5333.9 1695.76  5392.6 1694.18
  5425.3 1712.93  5465.2 1719.13  5510.7 1736.36  5546.5 1739.44    5559 1740.74
#Mann= 12 ,-1 , 0
    3937    .063       0  4004.1      .1       0  4085.1    .035       0
  4473.9      .1       0  4619.2    .063       0  4676.2    .035       0
  4841.8      .1       0  4982.3     .05       0  5013.1      .1       0
  5135.9     .07       0  5235.5    .094       0  5546.5      .1       0
Bank Sta=4982.3,5013.1
XS Rating Curve= 0 ,0
Exp/Cntr=0.3,0.1

Type RM Length L Ch R = 1 ,13366   ,583,583,583
BEGIN DESCRIPTION:
Town Creek 23.0
END DESCRIPTION:
XS GIS Cut Line= 3
      1922256.62     13939497.76        1921575.       13939025.
      1920714.24     13938609.32
#Sta/Elev= 30
  4170.5 1685.21  4177.9 1685.35  4276.8 1688.14  4365.8 1685.64    4508 1675.73
  4605.3 1673.13  4625.2 1673.14  4698.8 1672.24  4791.8 1663.65  4863.2 1661.73
  4899.8 1657.04  4936.5 1656.22  5001.4 1648.44  5001.9 1647.94  5032.4 1648.44
  5061.8 1651.08  5095.5 1650.38  5124.2 1656.68  5164.9 1671.28  5187.6 1671.84
  5224.9  1677.6  5303.5 1680.68  5588.6 1692.57  5727.9 1699.58  5761.3 1707.91
  5821.2 1705.69  5847.9 1707.27  5907.8 1713.73  5948.4 1722.59  5955.9 1724.43
#Mann= 14 ,-1 , 0
  4170.5     .07       0  4177.9      .1       0  4365.8     .07       0
    4508      .1       0  4605.3     .07       0  4625.2      .1       0
  4791.8    .035       0  4936.5     .07       0  5001.4     .05       0
  5032.4     .07       0  5124.2      .1       0  5303.5     .07       0
  5588.6    .035       0  5948.4      .1       0
Bank Sta=5001.4,5032.4
XS Rating Curve= 0 ,0
Exp/Cntr=0.3,0.1

Type RM Length L Ch R = 1 ,12783   ,290,290,290
BEGIN DESCRIPTION:
Town Creek 22.0
END DESCRIPTION:
XS GIS Cut Line= 3
      1922224.97     13938874.97        1921925.       13938575.
      1921211.79     13938535.99
#Sta/Elev= 30
  4570.9  1675.5  4607.4 1675.04    4737 1672.64  4762.1 1668.98  4813.4 1664.39
  4832.2 1663.81  4852.2 1661.08    4864  1660.3  4884.9    1657  4940.3 1653.25
  4976.4 1647.33  4982.8 1648.18  4983.1 1644.01  4983.6 1643.51  5014.1 1644.01
  5034.7 1647.76  5100.8 1647.83  5144.1 1654.25  5176.8 1660.61  5193.9 1662.06
  5271.9 1665.65  5294.7 1668.08  5406.4 1670.85  5461.3 1671.25  5476.3 1672.62
  5482.7 1672.16  5488.4 1673.31  5500.4 1672.36  5650.6 1678.81  5709.4 1683.31
#Mann= 7 ,-1 , 0
  4570.9     .07       0  4607.4      .1       0  4852.2    .035       0
  4983.1    .035       0  5014.1    .035       0  5144.1     .07       0
  5406.4    .035       0
Bank Sta=4983.1,5014.1
XS Rating Curve= 0 ,0
Exp/Cntr=0.3,0.1

Type RM Length L Ch R = 1 ,12493   ,257,257,257
BEGIN DESCRIPTION:
Town Creek 21.1
END DESCRIPTION:
XS GIS Cut Line= 4
      1923643.17     13938341.65      1922128.45     13938228.81
      1921889.73     13938337.32      1920926.17     13938454.51
#Sta/Elev= 30
  3292.7 1722.98  3340.6 1709.87  3424.7 1691.07  3435.8 1689.77  3493.9 1687.02
  3692.3 1684.23  4137.7 1676.07  4631.2 1672.01  4932.5 1670.39    4950 1667.29
  4969.7  1653.9  4976.3 1651.07  4977.1 1642.04  4977.7 1641.54  5010.3 1642.04
  5038.9 1645.95  5071.9 1648.28  5081.1 1647.08  5150.6 1649.66  5165.7 1649.88
  5177.8 1654.47  5211.1 1657.98  5353.1  1662.4  5389.4 1665.48  5622.1 1673.88
  5697.6 1678.17  5924.3 1698.95  5948.4 1703.15  5991.9 1705.39  6044.5 1709.16
#Mann= 7 ,-1 , 0
  3292.7      .1       0  3692.3     .07       0  4631.2      .1       0
  4977.1     .05       0  5010.3      .1       0  5150.6    .035       0
  5991.9    .094       0
Bank Sta=4977.1,5010.3
XS Rating Curve= 0 ,0
Exp/Cntr=0.3,0.1

Type RM Length L Ch R = 1 ,12236   ,542,542,542
BEGIN DESCRIPTION:
Town Creek 21.0
END DESCRIPTION:
XS GIS Cut Line= 4
      1923704.46     13938267.96      1922441.48     13937942.55
        1921775.       13938125.      1920975.05     13938324.99
#Sta/Elev= 30
  3004.5  1729.3  3048.8 1726.01  3120.7 1710.61  3154.2 1706.22  3194.1  1698.1
  3238.5 1692.91  3295.2 1688.62  3508.2 1684.93  4021.6 1674.81  4431.1 1670.33
  4808.2 1668.91  4950.1 1667.28  4962.9 1663.93  4965.9 1660.93  4970.8 1650.89
  4983.6 1641.29  4984.2 1640.79  5016.8 1641.29  5040.4 1645.29  5123.9 1648.41
  5136.3  1652.2  5170.3 1652.33    5292  1664.5  5640.3 1685.91  5717.7 1694.55
  5739.3 1695.12  5757.9 1698.93  5785.7 1699.27  5796.5  1702.8  5824.3 1705.07
#Mann= 7 ,-1 , 0
  3004.5      .1       0  3508.2     .07       0  4808.2      .1       0
  4950.1    .035       0  4983.6    .035       0  5016.8    .035       0
  5796.5    .094       0
Bank Sta=4983.6,5016.8
XS Rating Curve= 0 ,0
Exp/Cntr=0.3,0.1

Type RM Length L Ch R = 1 ,11694   ,368,368,368
BEGIN DESCRIPTION:
Town Creek 20.0
END DESCRIPTION:
XS GIS Cut Line= 4
      1923734.87     13938211.54      1922393.58     13937804.41
        1921525.       13937675.      1920924.99     13937424.99
#Sta/Elev= 30
  2720.1 1722.48  2809.8 1716.05  2906.5 1699.29  2981.7 1693.52    3249 1686.13
    4064 1671.62  4412.8 1664.42  4676.4 1663.81  4809.5    1664  4859.9 1659.34
  4917.7 1645.18  4941.8 1645.26    4954 1641.48  4987.1 1639.75  5005.5 1638.84
  5006.1 1638.34  5038.8 1638.84  5044.9 1643.27  5083.9 1647.11  5122.9 1663.58
  5165.2 1667.72  5261.6    1672  5327.7 1675.73  5360.2 1674.11  5460.7 1677.41
  5477.2 1680.56  5495.1 1688.02  5554.8 1704.64  5581.2 1714.85    5650 1725.49
#Mann= 10 ,-1 , 0
  2720.1      .1       0    3249     .07       0    4064      .1       0
  4412.8     .07       0  4676.4      .1       0  4859.9    .094       0
  4987.1     .07       0  5005.5     .05       0  5038.8     .07       0
  5261.6    .035       0
Bank Sta=5005.5,5038.8
XS Rating Curve= 0 ,0
Exp/Cntr=0.3,0.1

Type RM Length L Ch R = 1 ,11326   ,277,277,277
BEGIN DESCRIPTION:
Town Creek 19.1
END DESCRIPTION:
XS GIS Cut Line= 4
       1924542.1     13937187.23      1922142.13     13937266.54
      1921668.52      13937331.4      1920933.11     13937369.41
#Sta/Elev= 30
  1978.2 1784.86  2364.5 1750.23  2949.3 1715.06  3700.8 1688.16  3786.7 1679.75
  3876.8 1675.12  3953.5 1690.72  4032.9 1695.25  4074.9 1669.95    4135 1668.03
    4180 1672.86    4231 1666.17    4270 1678.22  4336.1 1681.65  4358.2 1678.29
  4387.2 1663.88  4409.2 1663.23    4637 1657.44  4703.6 1648.36  4726.3 1658.62
  4785.8 1659.79    4975 1639.18  4975.6 1638.68  5008.3 1639.18  5063.8 1642.94
  5105.1 1663.96  5118.8 1663.84  5400.2 1680.38  5517.4 1714.27  5593.9  1725.8
#Mann= 10 ,-1 , 0
  1978.2    .035       0  2364.5      .1       0  3700.8    .035       0
  3786.7    .063       0  3953.5    .035       0  4409.2      .1       0
  4785.8    .094       0    4975     .05       0  5008.3    .094       0
  5118.8    .035       0
Bank Sta=4975,5008.3
XS Rating Curve= 0 ,0
Exp/Cntr=0.3,0.1

Type RM Length L Ch R = 1 ,11049   ,425,425,425
BEGIN DESCRIPTION:
Town Creek 19.0
END DESCRIPTION:
XS GIS Cut Line= 3
      1922405.96     13936873.78      1921595.02     13937105.97
      1921215.73      13937097.6
#Sta/Elev= 30
  4136.2 1666.82  4259.4 1661.82  4543.4 1660.33  4587.1 1659.82  4608.9 1667.36
  4630.8 1666.89  4656.7 1660.29  4743.1 1656.88  4789.9 1649.86  4836.7 1647.69
  4855.4 1642.48  4861.5 1643.06  4924.1 1644.03  4930.3 1641.83  4945.9 1640.59
  4958.4  1642.9  4977.1 1640.15  4995.9 1641.11  5001.2 1640.45  5002.2 1637.47
  5002.9 1636.97  5036.2 1637.47  5061.3 1641.26  5076.3 1641.06    5085  1645.4
  5100.3 1653.74  5112.3 1653.79  5129.6 1658.33  5160.3 1662.41  5359.1 1665.46
#Mann= 6 ,-1 , 0
  4136.2    .063       0  4543.4    .035       0  4861.5    .094       0
  5002.2     .05       0  5036.2    .094       0    5085     .07       0
Bank Sta=5002.2,5036.2
XS Rating Curve= 0 ,0
Exp/Cntr=0.3,0.1

Type RM Length L Ch R = 1 ,10624   ,603,603,603
BEGIN DESCRIPTION:
Town Creek 18.0
END DESCRIPTION:
XS GIS Cut Line= 3
      1922548.41     13936812.06        1921625.       13936725.
      1920994.42     13936712.88
#Sta/Elev= 30
  4067.3 1675.43  4159.1 1676.92  4235.9 1668.15  4508.8 1660.53  4558.3 1661.25
  4582.5 1666.48  4586.3 1668.82  4600.6 1672.03  4639.7 1669.94  4668.5 1660.01
    4686 1659.77  4728.4 1659.85  4766.3 1658.79  4817.5 1649.79    4848  1646.9
  4895.9 1641.97    4932 1641.57    4946 1638.65  4950.1 1638.65  4951.1  1635.4
  4951.8  1634.9  4985.2  1635.4  5016.3  1635.9  5034.7 1639.12    5067  1643.5
  5090.5 1658.07  5105.2  1660.7  5370.4 1664.37  5574.4 1674.69  5625.5  1678.5
#Mann= 10 ,-1 , 0
  4067.3    .063       0  4586.3    .035       0    4686     .07       0
  4728.4    .035       0    4848    .094       0    4946    .035       0
  4951.1    .035       0  4985.2    .035       0  5034.7     .07       0
  5574.4      .1       0
Bank Sta=4951.1,4985.2
XS Rating Curve= 0 ,0
Exp/Cntr=0.3,0.1

Type RM Length L Ch R = 1 ,10021   ,519,519,519
BEGIN DESCRIPTION:
Town Creek 17.0
END DESCRIPTION:
XS GIS Cut Line= 3
      1922834.12     13936536.01      1921720.93     13936181.09
      1921075.01       13935975.
#Sta/Elev= 30
  3835.1 1690.84  3872.2 1688.29  3957.3 1687.29    3968 1687.74  4015.2 1682.36
  4120.5  1677.3  4213.6 1667.94  4256.6 1665.51    4434  1659.3  4764.6  1656.9
  4786.6 1655.62  4805.8 1649.62  4830.8 1645.04  4884.5 1639.17  4934.7 1637.66
  4967.8 1634.56  4968.5 1634.06  5001.9 1634.56  5003.9 1638.16  5029.1 1655.01
  5044.9 1659.36  5183.4  1658.1  5252.7 1654.89  5307.1 1657.55  5438.8 1657.88
  5463.7 1657.86  5545.6 1671.62  5615.1 1673.33  5648.5 1680.22  5681.5 1682.09
#Mann= 7 ,-1 , 0
  3835.1    .063       0  3957.3      .1       0  4256.6    .035       0
  4967.8    .035       0  5001.9    .035       0  5438.8    .063       0
  5648.5    .035       0
Bank Sta=4967.8,5001.9
XS Rating Curve= 0 ,0
Exp/Cntr=0.3,0.1

Type RM Length L Ch R = 1 ,9502    ,559,559,559
BEGIN DESCRIPTION:
Town Creek 16.0
END DESCRIPTION:
XS GIS Cut Line= 3
      1922806.15     13935883.93        1921825.       13935725.
      1921274.97     13935374.98
#Sta/Elev= 30
  4002.2 1677.79    4093 1675.15  4126.4 1675.54  4515.4 1661.86  4598.7  1660.8
  4727.4 1658.69  4859.7 1655.55    4899 1644.92  4924.7 1642.09    4947 1639.83
  4992.6 1639.75  5002.3  1637.6  5003.3 1634.09  5003.9 1633.59  5037.6 1634.09
  5040.9 1635.24  5123.5 1635.87  5144.9 1640.15  5169.6 1648.53  5208.4 1651.55
  5226.7 1652.08  5245.7 1649.24  5326.1 1653.84    5380 1653.28    5472 1653.69
  5543.1 1657.37  5564.5 1661.46  5614.3 1675.62  5627.6 1677.38  5648.1 1677.17
#Mann= 8 ,-1 , 0
  4002.2      .1       0  4598.7     .07       0  4727.4      .1       0
  4924.7    .035       0  5003.3    .035       0  5037.6    .035       0
  5208.4    .063       0    5380    .035       0
Bank Sta=5003.3,5037.6
XS Rating Curve= 0 ,0
Exp/Cntr=0.3,0.1

Type RM Length L Ch R = 1 ,8943    ,543,543,543
BEGIN DESCRIPTION:
Town Creek 15.0
END DESCRIPTION:
XS GIS Cut Line= 3
      1922843.37     13935363.93        1921725.       13935225.
      1921324.97       13935275.
#Sta/Elev= 30
  3877.3 1671.58    4123 1663.37  4135.3 1664.65  4172.9 1662.22  4204.7 1662.72
    4253 1656.21    4259  1660.1    4270 1660.57  4361.9 1659.12  4373.9 1656.22
    4386 1659.29  4422.3 1656.44  4500.8  1657.1  4522.1  1654.7  4600.2 1653.63
  4816.7  1652.5  4911.6 1648.92  4930.7 1640.87  4942.3 1636.99  4960.4 1634.61
  4986.6 1634.17  4987.3 1633.67    5021 1634.17  5066.2 1637.47  5105.5 1643.05
  5162.7 1647.92    5314  1653.9  5329.3 1656.58  5377.6 1669.91  5407.4 1673.36
#Mann= 8 ,-1 , 0
  3877.3      .1       0    4270     .07       0  4600.2      .1       0
  4816.7    .035       0  4930.7      .1       0  4986.6     .05       0
    5021      .1       0    5314    .035       0
Bank Sta=4986.6,5021
XS Rating Curve= 0 ,0
Exp/Cntr=0.3,0.1

Type RM Length L Ch R = 1 ,8400    ,528,528,528
BEGIN DESCRIPTION:
Town Creek 14.0
END DESCRIPTION:
XS GIS Cut Line= 3
       1922578.6      13934901.4        1921625.       13934775.
      1921225.04       13934775.
#Sta/Elev= 30
    4043 1660.79    4143 1656.33    4338 1652.09  4345.7  1651.5  4357.8 1647.41
    4376 1651.73    4471 1651.33  4575.7  1648.5  4603.3 1649.11  4702.3 1649.07
  4796.6    1651    4836 1648.64  4865.7 1650.41  4881.4  1650.1  4902.5 1638.86
  4908.6 1637.01  4952.8 1636.21  4954.8    1634  4955.5  1633.5  4989.4    1634
  5053.4 1634.87  5077.4  1640.1  5098.1    1643  5134.4 1648.36  5182.4 1662.73
  5209.6 1664.87  5238.4 1666.37  5290.4 1665.49  5326.4 1666.99  5404.9 1666.75
#Mann= 9 ,-1 , 0
    4043      .1       0    4471     .07       0  4603.3      .1       0
  4702.3    .035       0  4865.7      .1       0  4954.8     .05       0
  4989.4      .1       0  5098.1    .035       0  5209.6    .063       0
Bank Sta=4954.8,4989.4
XS Rating Curve= 0 ,0
Exp/Cntr=0.3,0.1

Type RM Length L Ch R = 1 ,7872    ,1102,1102,1102
BEGIN DESCRIPTION:
Town Creek 13.0
END DESCRIPTION:
XS GIS Cut Line= 3
      1922533.97     13934811.02        1921725.       13934325.
      1920993.52     13934248.61
#Sta/Elev= 30
  4056.3 1659.31  4389.1 1648.25  4406.8 1647.13  4424.3 1648.45  4438.3 1640.91
  4441.8 1641.49  4448.7 1647.27  4482.6 1647.03  4734.8 1644.89  4795.3 1645.01
  4866.3 1640.93  4889.8 1642.08  4914.4 1637.84  4942.8  1630.5  4971.3 1630.77
  4984.3 1626.07    4996 1624.66  4996.7 1624.16  5030.6 1624.66  5031.7 1630.59
  5037.8 1632.03  5079.9 1633.92    5095 1636.05  5128.2 1646.45  5179.2 1650.44
  5191.7 1650.49  5438.9 1651.99  5514.3 1654.74  5625.9 1653.62  5735.5 1656.31
#Mann= 9 ,-1 , 0
  4056.3      .1       0  4389.1     .07       0  4482.6      .1       0
  4734.8    .035       0    4996    .035       0  5030.6    .035       0
  5079.9    .063       0  5179.2    .094       0  5191.7    .063       0
Bank Sta=4996,5030.6
XS Rating Curve= 0 ,0
Exp/Cntr=0.3,0.1

Type RM Length L Ch R = 1 ,6770    ,569,569,569
BEGIN DESCRIPTION:
Town Creek 12.0
END DESCRIPTION:
XS GIS Cut Line= 4
        1923075.       13934175.        1922575.       13933925.
      1921876.93     13933725.83      1920999.41     13933753.46
#Sta/Elev= 30
    4441 1750.17  4476.2 1747.46  4496.5 1743.22  4509.7 1737.33  4543.3 1730.12
  4559.1 1722.77  4576.8 1716.46  4610.6 1712.75  4671.4 1687.88  4751.2  1659.4
  4811.8 1649.18  4855.2 1639.04    4929 1634.37  4935.7 1632.27  4942.4 1624.92
  4962.1 1620.29  4962.8 1619.79  4996.9 1620.29    5000  1624.6    5059 1624.75
  5099.5 1637.42  5130.7 1642.88  5242.2 1644.96  5623.4 1645.51  5840.5  1643.6
  5868.7 1644.17  6037.9 1644.51  6052.7 1644.62  6104.8 1646.17  6603.9 1643.78
#Mann= 10 ,-1 , 0
    4441      .1       0  4559.1    .035       0  4962.1    .035       0
  4996.9    .035       0  5242.2    .063       0  5623.4    .035       0
  5840.5    .063       0  5868.7    .035       0  6037.9    .063       0
  6052.7    .035       0
Bank Sta=4962.1,4996.9
XS Rating Curve= 0 ,0
Exp/Cntr=0.3,0.1

Type RM Length L Ch R = 1 ,6201    ,521,521,521
BEGIN DESCRIPTION:
Town Creek 11.0
END DESCRIPTION:
XS GIS Cut Line= 3
      1923075.01       13933475.        1922675.       13933425.
      1921825.31     13933652.74
#Sta/Elev= 30
  4602.3 1684.33  4652.4 1681.49  4685.7 1672.47    4728 1667.05  4763.2 1656.03
  4783.2 1653.66  4812.6 1649.32  4845.9 1647.25    4864 1644.42  4888.2 1644.83
  4903.8 1638.82  4927.5 1634.75  4939.4 1628.51  4960.8 1623.14  4961.5 1620.17
  4962.2 1619.67  4996.4 1620.17    4997 1621.52  5006.1 1623.17    5073 1628.34
    5085 1628.18  5124.2 1628.65  5152.1 1632.61    5171 1638.95  5193.4 1640.49
  5270.1 1642.58    5425 1642.23  5528.1 1643.91  5666.9 1643.63  5885.1 1643.03
#Mann= 9 ,-1 , 0
  4602.3    .035       0  4783.2    .063       0  4939.4    .035       0
  4961.5    .035       0  4996.4    .035       0    5085    .063       0
  5193.4    .035       0  5528.1    .063       0  5666.9    .035       0
Bank Sta=4961.5,4996.4
XS Rating Curve= 0 ,0
Exp/Cntr=0.3,0.1

Type RM Length L Ch R = 1 ,5680    ,635,635,635
BEGIN DESCRIPTION:
Town Creek 10.0
END DESCRIPTION:
XS GIS Cut Line= 3
      1922606.95     13932732.76      1922380.16     13933017.72
      1921659.08     13933596.45
#Sta/Elev= 30
  4626.7 1651.15    4692 1647.44  4754.6 1645.39  4761.3 1643.11  4777.6 1642.23
  4907.8 1643.75  4923.2 1635.51  4933.8 1623.63  4941.5 1618.55  4956.8 1618.56
  4958.7 1617.33  4959.5 1616.83  4993.8 1617.33  4994.6 1618.73  4998.4 1619.43
  5020.2 1618.65  5025.3 1619.72  5065.7 1621.09  5090.7 1624.78  5117.7 1624.86
  5152.3 1630.17  5279.2 1636.56    5378 1638.21  5456.2 1638.43    5531 1640.47
    5560 1639.59  5617.7 1641.67  5765.2 1642.11  5874.7 1642.79  5915.5 1643.28
#Mann= 6 ,-1 , 0
  4626.7    .035       0  4958.7    .035       0  4993.8    .035       0
    5378    .063       0  5765.2    .035       0  5874.7    .063       0
Bank Sta=4958.7,4993.8
XS Rating Curve= 0 ,0
Exp/Cntr=0.3,0.1

Type RM Length L Ch R = 1 ,5045    ,546,546,546
BEGIN DESCRIPTION:
Town Creek 9.0
END DESCRIPTION:
XS GIS Cut Line= 3
      1922351.73     13932365.31        1921875.       13932725.
      1921454.94     13933498.39
#Sta/Elev= 30
  4402.8 1657.05    4476 1658.61  4505.3 1657.18  4517.3 1658.79  4562.7 1657.51
    4600 1656.41  4618.8 1653.75  4712.8 1649.25  4722.1 1647.36  4791.7 1643.44
  4951.3 1638.94  4963.6 1633.91  4968.3 1626.82  4974.8 1622.36  4978.5 1618.09
  4984.8 1614.65  4985.6 1614.15  5019.9 1614.65  5022.7 1617.14  5029.7 1618.02
  5055.9 1617.01  5104.8 1618.74  5132.1 1622.49  5191.8 1626.47    5255 1631.68
    5354 1636.69  5450.5 1637.45    5597 1639.28  5679.3 1640.05  5880.1  1642.9
#Mann= 8 ,-1 , 0
  4402.8    .063       0  4562.7    .035       0  4984.8    .035       0
  5019.9    .035       0  5191.8    .063       0  5450.5    .035       0
    5597    .063       0  5679.3    .035       0
Bank Sta=4984.8,5019.9
XS Rating Curve= 0 ,0
Exp/Cntr=0.3,0.1
