HEC-RAS study Turtle Creek.prj: Turtle Creek Base Level Engineering

--- Turtle Creek.g01 (geometry) --- (continued)

Type RM Length L Ch R = 1 ,97527   ,266,266,266
BEGIN DESCRIPTION:
Mapping XS a9e2248b
END DESCRIPTION:
XS GIS Cut Line= 3
      1886780.29      13907279.2      1886931.35     13906888.14
      1886975.98     13906268.86
#Sta/Elev= 30
  4517.7 1954.02    4596 1947.79  4640.1 1941.22  4725.9 1935.67  4735.1 1927.49
  4740.4 1924.66    4758  1893.6    4765 1884.88  4770.4 1884.17  4789.6 1875.95
    4800 1873.33  4833.1 1867.11  4874.1 1865.53  4904.1 1866.64    4990 1857.89
  4990.5 1857.39  5010.5 1857.89  5040.3 1859.95  5056.3 1864.87  5110.5 1866.24
  5170.7 1872.87  5201.1 1873.27  5240.8 1889.37  5273.4 1899.17    5291 1903.61
  5335.8  1911.1  5341.1 1913.61  5431.3 1932.49  5461.4 1937.49  5557.8 1942.39
#Mann= 5 ,-1 , 0
  4517.7      .1       0    4800     .07       0    4990     .05       0
  5010.5     .07       0  5273.4      .1       0
Bank Sta=4990,5010.5
XS Rating Curve= 0 ,0
Exp/Cntr=0.3,0.1

Type RM Length L Ch R = 1 ,97261   ,393,393,393
BEGIN DESCRIPTION:
Turtle Creek 159.0
END DESCRIPTION:
XS GIS Cut Line= 4
      1887374.99     13907224.98      1887185.32     13906959.44
      1887180.75     13906777.43      1887324.99     13906525.02
#Sta/Elev= 30
  4589.2 1936.05  4667.8 1921.95  4682.6 1917.68  4718.2 1913.92    4733 1908.87
  4753.8 1906.72  4783.3 1899.89  4860.8 1889.67  4875.5 1879.54  4884.1 1866.28
    4929 1863.17    4940 1864.26    4980 1857.82    4990 1859.22  5016.8 1857.89
  5019.6 1857.63  5020.1 1857.13  5040.3 1857.63    5090 1862.86  5117.6 1863.51
  5160.3 1864.88    5204 1865.09  5213.4 1870.55  5219.2 1871.55    5235 1884.06
  5240.8 1885.83  5256.6  1896.1  5307.7 1911.36  5337.2 1915.33  5388.3 1917.55
#Mann= 7 ,-1 , 0
  4589.2      .1       0    4929     .07       0  5016.8      .1       0
  5019.6     .05       0  5040.3      .1       0  5117.6     .07       0
  5160.3      .1       0
Bank Sta=5019.6,5040.3
XS Rating Curve= 0 ,0
Exp/Cntr=0.3,0.1

Type RM Length L Ch R = 1 ,96868   ,131,131,131
BEGIN DESCRIPTION:
Mapping XS ef71124f
END DESCRIPTION:
XS GIS Cut Line= 2
       1887643.9     13907241.96      1887443.12     13906481.52
#Sta/Elev= 30
    4672 1965.42  4731.3 1961.58  4751.6 1957.37  4761.2 1949.69  4766.4 1949.77
  4772.3 1945.28  4887.2 1908.28  4922.3 1892.66  4927.5 1892.42  4957.4 1881.38
  4962.6 1881.09  4979.1 1870.83  4982.9 1866.34  4989.5 1858.55  4999.8 1850.82
  5000.3 1850.32  5020.5 1850.82  5078.2 1858.35  5123.9 1858.79    5186 1855.47
  5206.1 1861.91    5217 1864.02    5248  1863.2  5258.4 1865.47  5279.5 1877.01
  5299.8 1892.15  5322.1 1901.32  5361.8 1905.56  5430.3 1908.62  5458.5 1912.21
#Mann= 6 ,-1 , 0
    4672      .1       0  4982.9    .035       0  4999.8    .035       0
  5020.5    .035       0  5206.1     .07       0  5322.1      .1       0
Bank Sta=4999.8,5020.5
XS Rating Curve= 0 ,0
Exp/Cntr=0.3,0.1

Type RM Length L Ch R = 1 ,96737   ,569,569,569
BEGIN DESCRIPTION:
Turtle Creek 158.0
END DESCRIPTION:
XS GIS Cut Line= 3
      1887975.01     13907175.01        1887675.       13906875.
        1887575.     13906474.99
#Sta/Elev= 30
  4575.4 1993.73    4632 1981.37  4688.6 1973.07    4731 1962.94  4759.3 1948.08
  4787.5 1935.37  4801.7 1924.89  4886.5 1888.55  4943.1 1869.54  4964.3 1855.99
  4971.4 1850.49  4985.7 1850.37  4986.2 1849.87  5006.5 1850.37  5017.7 1855.73
  5030.6 1857.51  5064.1 1858.17  5113.1 1854.48  5146.6 1856.57  5179.2 1862.69
    5229 1864.82  5247.1 1871.58  5257.4 1877.24  5265.1 1885.12  5270.3 1888.47
  5290.9 1897.31  5306.3 1901.83  5352.7 1905.88  5388.8 1913.82    5412 1914.49
#Mann= 6 ,-1 , 0
  4575.4      .1       0  4964.3    .035       0  4985.7    .035       0
  5006.5    .035       0  5179.2     .07       0  5290.9      .1       0
Bank Sta=4985.7,5006.5
XS Rating Curve= 0 ,0
Exp/Cntr=0.3,0.1

Type RM Length L Ch R = 1 ,96168   ,542,542,542
BEGIN DESCRIPTION:
Turtle Creek 157.0
END DESCRIPTION:
XS GIS Cut Line= 3
        1888175.     13907074.97        1888175.       13906675.
      1887824.98     13906224.97
#Sta/Elev= 30
  4605.1 1992.14  4645.1 1983.03  4695.1 1976.88  4735.1 1966.17  4805.1 1958.03
  4845.1 1945.08  4875.1 1939.09  4885.1 1933.21  4895.1 1923.25  4925.1 1906.72
  4935.1 1907.95  4945.1 1902.04  4965.1 1883.52  4975.1 1851.43  5001.9 1848.69
  5002.4 1848.19  5022.7 1848.69  5041.3 1849.26  5076.6 1855.11  5225.9 1859.31
  5265.7 1862.94  5296.5 1862.31  5319.1 1867.76  5339.9 1875.59  5350.6 1875.32
  5375.2 1876.59  5389.7 1890.37  5410.5 1897.89  5492.6 1916.77  5575.2 1932.21
#Mann= 6 ,-1 , 0
  4605.1      .1       0  5001.9     .05       0  5022.7      .1       0
  5265.7      .1       0  5350.6     .07       0  5492.6      .1       0
Bank Sta=5001.9,5022.7
XS Rating Curve= 0 ,0
Exp/Cntr=0.3,0.1

Type RM Length L Ch R = 1 ,95626   ,529,529,529
BEGIN DESCRIPTION:
Turtle Creek 156.0
END DESCRIPTION:
XS GIS Cut Line= 3
        1888775.     13906725.01        1888575.       13906375.
      1887925.04     13906125.01
#Sta/Elev= 30
  4593.5 1948.51    4623 1945.12  4674.1    1943  4725.2    1937  4741.1  1931.5
  4784.3 1922.37  4908.1 1908.28  4984.5 1895.62  4988.7 1894.38  4993.7 1872.92
  4999.3 1872.92  5001.2 1848.15  5001.7 1847.65    5022 1848.15  5041.6 1849.46
  5120.9 1848.18  5157.3 1850.25  5230.2 1850.82  5265.5 1855.53  5284.8  1855.3
  5314.8 1861.39  5367.2 1862.61  5429.5  1865.9  5454.1 1865.21  5459.5 1866.88
  5485.2 1881.56  5553.8 1905.37  5585.9 1910.14    5618 1917.35    5693 1927.88
#Mann= 6 ,-1 , 0
  4593.5      .1       0  4984.5     .07       0  5001.2     .05       0
    5022     .07       0  5367.2     .07       0  5485.2      .1       0
Bank Sta=5001.2,5022
XS Rating Curve= 0 ,0
Exp/Cntr=0.3,0.1

Type RM Length L Ch R = 1 ,95097   ,561,561,561
BEGIN DESCRIPTION:
Turtle Creek 155.0
END DESCRIPTION:
XS GIS Cut Line= 3
      1889175.01     13906875.01        1888875.       13906075.
      1888724.99     13905624.96
#Sta/Elev= 30
  4150.1 2001.84  4182.2 1996.58  4220.4 1986.29  4267.6 1979.73  4305.9 1969.59
  4342.4 1964.49  4391.3 1952.19  4470.5 1942.36  4531.9 1925.26  4662.8 1905.04
  4702.8 1893.09  4763.3 1892.17  4812.3 1885.46  4848.8  1876.7  4933.5 1849.84
  4991.1 1845.66  4991.6 1845.16  5012.5 1845.66  5046.7 1846.24  5078.3 1849.06
  5088.8 1852.11  5160.4 1853.51  5265.2 1857.25  5331.3 1860.84  5362.9 1875.78
  5394.5 1903.14  5405.1 1909.85  5426.2 1916.95  5436.7 1923.59  5478.9 1925.92
#Mann= 6 ,-1 , 0
  4150.1      .1       0  4933.5     .07       0  4991.1     .05       0
  5012.5     .07       0  5160.4      .1       0  5265.2     .07       0
Bank Sta=4991.1,5012.5
XS Rating Curve= 0 ,0
Exp/Cntr=0.3,0.1

Type RM Length L Ch R = 1 ,94536   ,506,506,506
BEGIN DESCRIPTION:
Turtle Creek 154.0
END DESCRIPTION:
XS GIS Cut Line= 3
      1889825.01     13906475.02        1889325.       13905775.
      1889124.98     13905424.97
#Sta/Elev= 30
  4144.2 1969.99  4193.4 1965.21  4253.2 1951.54  4316.3  1944.2    4374 1919.97
  4430.6 1901.62  4460.1 1887.87  4480.9 1883.58  4495.7 1876.12  4546.1 1862.61
  4581.7 1858.83  4657.8 1858.68  4669.3 1857.38  4760.3 1853.69  4860.7 1849.23
  4882.2 1844.51  4986.4 1842.18  4986.9 1841.68  5007.8 1842.18  5136.2 1850.04
  5157.8 1856.95  5186.3 1873.86  5195.2 1881.89  5211.1 1891.18  5216.8 1890.75
  5223.3 1907.62  5232.6 1914.57  5281.6 1919.18  5400.9  1920.8  5407.6 1920.88
#Mann= 10 ,-1 , 0
  4144.2     .07       0  4253.2      .1       0  4657.8    .035       0
  4669.3     .07       0  4760.3    .035       0  4882.2     .07       0
  4986.4     .05       0  5007.8     .07       0  5186.3      .1       0
  5400.9     .07       0
Bank Sta=4986.4,5007.8
XS Rating Curve= 0 ,0
Exp/Cntr=0.3,0.1

Type RM Length L Ch R = 1 ,94030   ,574,574,574
BEGIN DESCRIPTION:
Turtle Creek 153.0
END DESCRIPTION:
XS GIS Cut Line= 3
      1890175.02     13906075.02        1889775.       13905775.
        1889475.       13905475.
#Sta/Elev= 30
  4495.5 1948.92  4523.7 1944.66  4538.2  1934.3    4582 1908.04  4595.5 1895.08
  4609.1 1885.54  4617.4 1882.02  4624.6 1876.75  4638.2 1868.57  4659.1  1858.9
  4673.7 1854.43  4688.2 1852.54  4773.7 1850.89  4859.1 1852.17  4873.7 1850.32
  4888.2 1846.65  4923.7 1842.71  5013.1 1839.91  5013.6 1839.41  5034.5 1839.91
  5046.8 1842.47  5066.2 1845.96  5108.7 1846.49  5122.8 1848.71    5137 1855.45
  5151.1 1867.08  5165.2 1897.16  5193.5 1900.68  5250.1 1904.79  5419.8 1906.42
#Mann= 5 ,-1 , 0
  4495.5      .1       0  4624.6     .07       0  5013.1     .05       0
  5034.5     .07       0  5046.8      .1       0
Bank Sta=5013.1,5034.5
XS Rating Curve= 0 ,0
Exp/Cntr=0.3,0.1

Type RM Length L Ch R = 1 ,93456   ,555,555,555
BEGIN DESCRIPTION:
Turtle Creek 152.0
END DESCRIPTION:
XS GIS Cut Line= 3
        1890275.     13905975.03        1890275.       13905575.
      1889724.95     13905474.99
#Sta/Elev= 30
    4600 1949.53    4640  1947.9    4660  1942.2    4700 1927.77    4710 1925.44
    4750 1907.73    4770 1887.13    4780 1883.86    4840    1858    4870 1847.08
    4880 1843.87    4890 1842.33  4902.4 1842.18    4950 1839.48  4969.3 1834.91
  4969.8 1834.41  4990.8 1834.91    5122 1840.86  5172.8 1847.08  5203.3 1847.23
    5317  1851.5  5396.4 1854.84  5420.6 1860.53  5426.9 1863.84  5467.6 1876.25
  5473.9 1879.52    5479 1879.86  5508.2 1889.02  5527.3 1892.89  5559.1 1894.82
#Mann= 5 ,-1 , 0
    4600      .1       0  4902.4     .07       0  4969.3     .05       0
  4990.8     .07       0    5317      .1       0
Bank Sta=4969.3,4990.8
XS Rating Curve= 0 ,0
Exp/Cntr=0.3,0.1

Type RM Length L Ch R = 1 ,92901   ,362,362,362
BEGIN DESCRIPTION:
Turtle Creek 151.0
END DESCRIPTION:
XS GIS Cut Line= 3
      1890670.68     13905076.95        1890325.       13905075.
      1889724.96       13905125.
#Sta/Elev= 30
  4658.9 1904.01  4674.6 1906.02  4744.6 1910.25  4812.9 1912.33  4844.6 1912.61
  4884.6 1911.32  4894.6 1909.88  4904.6 1891.13  4914.6 1852.85  4924.6 1837.85
  4930.8 1836.04  4944.6 1833.51  4983.8 1833.32  4984.3 1832.82  5005.3 1833.32
  5014.6 1835.02  5044.7 1837.06  5062.3 1840.71  5074.8  1840.9  5104.9 1844.75
  5155.1 1846.56  5283.2 1846.65  5335.7 1847.01  5428.5  1851.1  5496.3 1866.38
  5536.4 1877.39  5543.9 1880.82  5556.5 1884.45  5596.6 1891.98  5606.7 1892.74
#Mann= 6 ,-1 , 0
  4658.9     .07       0  4812.9      .1       0  4930.8     .07       0
  4983.8     .05       0  5005.3     .07       0  5283.2      .1       0
Bank Sta=4983.8,5005.3
XS Rating Curve= 0 ,0
Exp/Cntr=0.3,0.1

Type RM Length L Ch R = 1 ,92539   ,190,190,190
BEGIN DESCRIPTION:
Turtle Creek 150.1
END DESCRIPTION:
XS GIS Cut Line= 4
      1890614.27     13904663.76      1890312.58     13904715.85
      1890258.32     13904733.22      1889715.81      13904893.8
#Sta/Elev= 30
  4706.9 1892.46  4747.7 1896.79    4814 1897.91    4917 1901.86  4929.4 1901.78
  4949.7 1898.11  4959.9 1893.64    4970 1867.43  4976.9 1854.92  4981.9 1852.45
  5000.4 1835.01  5013.1 1834.36  5015.7  1828.7  5016.2  1828.2  5037.2  1828.7
    5042 1832.88  5052.5 1829.45  5058.6 1829.67  5063.9 1833.16  5069.2 1832.09
  5091.5 1831.13  5096.7 1834.55  5218.2 1842.89  5380.6 1845.34  5438.5 1846.95
  5484.4 1851.45    5550  1864.5  5571.5 1866.63  5604.9 1872.93  5635.8 1878.39
#Mann= 10 ,-1 , 0
  4706.9     .07       0    4814      .1       0  5015.7     .05       0
  5037.2      .1       0  5069.2    .035       0  5218.2     .07       0
  5380.6      .1       0  5484.4     .07       0  5571.5      .1       0
  5604.9     .07       0
Bank Sta=5015.7,5037.2
XS Rating Curve= 0 ,0
Exp/Cntr=0.3,0.1

Type RM Length L Ch R = 1 ,92349   ,681,681,681
BEGIN DESCRIPTION:
Turtle Creek 150.0
END DESCRIPTION:
XS GIS Cut Line= 3
      1890575.03     13904374.98        1890225.       13904575.
      1889458.88     13904905.72
#Sta/Elev= 30
  4602.8 1899.27  4680.8 1897.28  4815.2 1896.12  4858.4 1890.58  4874.2 1880.78
    4880 1881.71  4890.1 1874.18  4895.8 1873.15  4902.3 1863.72  4911.6 1855.74
  4917.4 1855.72  4933.2 1844.13    4939 1844.25  4948.4  1833.3    4960 1828.71
  4987.3 1827.77  4987.8 1827.27  5008.8 1827.77  5052.4 1833.86  5071.6 1835.44
  5180.5 1842.14  5398.2 1847.44  5507.1 1861.59  5675.2 1886.23  5704.1 1889.23
  5722.2 1886.82  5727.6  1890.9  5745.7 1888.33  5768.4 1894.47  5840.4 1900.84
#Mann= 10 ,-1 , 0
  4602.8     .07       0  4680.8      .1       0    4960    .035       0
  4987.3    .035       0  5008.8    .035       0  5052.4     .07       0
  5071.6    .035       0  5180.5     .07       0  5398.2      .1       0
  5507.1     .07       0
Bank Sta=4987.3,5008.8
XS Rating Curve= 0 ,0
Exp/Cntr=0.3,0.1

Type RM Length L Ch R = 1 ,91668   ,423,423,423
BEGIN DESCRIPTION:
Turtle Creek 149.0
END DESCRIPTION:
XS GIS Cut Line= 3
        1890475.       13904325.      1890025.83     13904003.12
      1889674.96     13903824.98
#Sta/Elev= 30
  4445.9 1897.38  4488.9 1894.03  4509.8 1888.77  4574.9 1868.72  4625.2 1849.19
  4654.7 1841.89  4681.7 1839.29  4782.4 1837.56  4797.2 1833.47  4871.5 1830.31
  4897.9 1826.51  4948.3 1827.27  4979.2 1822.28  4979.7 1821.78  5000.9 1822.28
  5001.8 1825.43  5005.2 1827.24  5010.8 1827.74  5033.1 1838.52  5061.3 1838.83
  5116.5 1844.98    5161 1869.57  5183.3 1885.23  5190.1 1892.96  5227.8 1914.62
  5257.4    1936    5289 1952.83  5339.1 1986.05  5361.4 1991.53    5392 1992.57
#Mann= 5 ,-1 , 0
  4445.9      .1       0  4871.5     .07       0  4979.2     .05       0
  5000.9     .07       0  5061.3      .1       0
Bank Sta=4979.2,5000.9
XS Rating Curve= 0 ,0
Exp/Cntr=0.3,0.1

Type RM Length L Ch R = 1 ,91245   ,545,545,545
BEGIN DESCRIPTION:
Turtle Creek 148.0
END DESCRIPTION:
XS GIS Cut Line= 3
      1890525.02     13904225.04        1890225.       13903675.
      1889874.96     13903474.98
#Sta/Elev= 30
  4364.8 1898.85  4387.6 1895.86  4470.3 1869.95  4498.2 1862.34  4507.2  1850.1
    4520 1845.02  4579.8 1845.62  4644.3 1840.81  4688.3 1840.34  4911.6 1835.97
  4983.3 1825.68  4991.3 1823.78  4994.2 1819.24  4994.7 1818.74  5015.9 1819.24
  5042.5    1820  5079.9 1830.42  5085.6 1842.57  5101.5 1860.81  5107.2 1895.67
  5144.7 1927.32  5197.9 1953.47  5219.5 1967.55  5225.3 1980.22  5241.1 1987.98
  5246.9 1998.24  5250.5 2000.39  5268.5 2006.43  5327.5 2017.01  5394.5 2022.94
#Mann= 6 ,-1 , 0
  4364.8      .1       0  4470.3     .07       0  4644.3      .1       0
  4688.3     .07       0  4994.2     .05       0  5015.9      .1       0
Bank Sta=4994.2,5015.9
XS Rating Curve= 0 ,0
Exp/Cntr=0.3,0.1

Type RM Length L Ch R = 1 ,90700   ,579,579,579
BEGIN DESCRIPTION:
Turtle Creek 147.0
END DESCRIPTION:
XS GIS Cut Line= 3
        1890575.     13904225.01        1890675.       13903475.
      1890775.01     13903074.96
#Sta/Elev= 30
  4248.8  1899.8  4329.5 1886.78    4380 1873.77  4441.7 1863.82  4450.6 1861.77
  4460.7 1855.57  4490.9 1855.96  4541.4 1845.44  4581.7 1841.04  4672.9 1836.91
  4753.2 1835.47  4833.9 1838.08  4884.4 1837.38  4895.1 1835.47  4944.1 1817.23
  4944.6 1816.73  4965.9 1817.23  5037.7 1818.65    5057 1820.23  5064.7 1826.05
  5087.9 1829.78  5098.2 1834.68  5105.9 1841.67  5111.1 1840.14  5118.8 1848.45
  5139.4 1864.68  5147.2 1908.81  5201.3  1926.8  5345.6 1957.26  5417.8 1974.73
#Mann= 6 ,-1 , 0
  4248.8     .07       0  4672.9      .1       0  4895.1     .07       0
  4944.1     .05       0  4965.9     .07       0  5037.7      .1       0
Bank Sta=4944.1,4965.9
XS Rating Curve= 0 ,0
Exp/Cntr=0.3,0.1

Type RM Length L Ch R = 1 ,90121   ,409,409,409
BEGIN DESCRIPTION:
Turtle Creek 146.0
END DESCRIPTION:
XS GIS Cut Line= 3
      1890775.01     13904174.98        1891175.       13903575.
        1891375.       13903225.
#Sta/Elev= 30
  4284.4 1888.16  4312.9 1886.11    4385 1870.44  4415.1 1868.97  4457.1 1862.63
  4508.2 1849.09  4580.3 1839.73  4664.3 1835.24  4910.8 1829.98  4940.9 1827.88
  4976.9 1818.65  5002.5 1817.08    5003 1816.58  5024.3 1817.08  5041.5 1817.54
  5063.1 1817.73  5086.1 1828.96    5094 1831.08  5099.8 1829.34  5109.1 1833.11
  5115.6 1839.44  5121.4 1840.95  5131.5 1849.88  5137.2 1861.24  5143.7 1919.62
  5196.2 1944.69  5255.3 1970.32  5276.9 1977.75  5304.9 1980.52  5408.6 1984.15
#Mann= 5 ,-1 , 0
  4284.4     .07       0  4664.3    .035       0  5002.5    .035       0
  5024.3    .035       0  5041.5      .1       0
Bank Sta=5002.5,5024.3
XS Rating Curve= 0 ,0
Exp/Cntr=0.3,0.1

Type RM Length L Ch R = 1 ,89712   ,696,696,696
BEGIN DESCRIPTION:
Turtle Creek 145.0
END DESCRIPTION:
XS GIS Cut Line= 3
      1890875.01     13904274.99      1891470.12     13903819.62
      1891575.01     13903524.98
#Sta/Elev= 30
  4250.8 1887.36  4293.4 1883.05  4322.4 1874.49  4343.3 1874.32  4364.1 1870.88
  4486.6 1859.58  4607.1 1834.56  4742.8 1829.73  4800.4 1828.58    4871 1826.77
  4955.8  1817.9  4994.3 1817.45  4994.8 1816.95  5016.1 1817.45  5047.5 1819.35
  5056.1 1822.21  5079.4 1841.83    5087 1845.87  5092.3 1856.46  5111.2 1867.56
  5117.8 1894.24  5123.1 1898.79    5143 1906.85  5148.6 1910.91  5174.1  1918.1
  5185.5 1923.49    5205 1928.11  5266.6 1938.04  5271.9  1937.1  5312.9 1940.76
#Mann= 6 ,-1 , 0
  4250.8     .07       0  4742.8    .035       0  4800.4     .07       0
  4955.8      .1       0  4994.3     .05       0  5016.1      .1       0
Bank Sta=4994.3,5016.1
XS Rating Curve= 0 ,0
Exp/Cntr=0.3,0.1

Type RM Length L Ch R = 1 ,89016   ,302,302,302
BEGIN DESCRIPTION:
Turtle Creek 144.0
END DESCRIPTION:
XS GIS Cut Line= 3
      1890974.99       13904375.        1891775.       13904375.
      1892124.98     13904574.99
#Sta/Elev= 30
    4199 1875.49    4239 1873.19  4284.9 1866.45    4329 1862.24    4419 1847.29
    4479 1841.48    4509 1835.71  4699.1 1825.93    4789  1825.1    4809 1818.22
    4819 1817.48  4973.1 1817.41    4996  1817.4  4996.5  1816.9  5017.9  1817.4
  5050.1 1819.82  5055.1 1827.12    5066 1836.02  5071.7 1836.73  5087.6 1849.86
  5102.7 1857.22  5109.1 1864.77  5114.9 1866.76  5130.7 1903.93  5137.2 1921.41
  5189.8 1944.63  5224.7 1953.75  5286.2 1962.44  5356.8 1976.38  5402.1 1977.09
#Mann= 8 ,-1 , 0
    4199     .07       0  4284.9    .035       0  4699.1     .07       0
  4973.1    .033       0    4996    .033       0  5017.9    .033       0
  5055.1      .1       0  5224.7     .07       0
Bank Sta=4996,5017.9
XS Rating Curve= 0 ,0
Exp/Cntr=0.3,0.1

Type RM Length L Ch R = 1 ,88714   ,250,250,250
BEGIN DESCRIPTION:
Turtle Creek 143.1
END DESCRIPTION:
XS GIS Cut Line= 4
      1890946.24     13904492.33      1891623.34      13904639.9
      1891770.91     13904655.09      1892139.85     13904670.28
#Sta/Elev= 30
  4255.5 1884.46  4290.8 1876.05  4346.3 1872.86  4383.8 1867.74  4432.9 1866.92
  4438.5 1864.32    4541  1849.7    4575 1844.59  4612.5  1835.3  4673.9 1828.87
  4801.1 1823.62  4814.9 1823.35  4919.5 1824.37  4960.2  1821.7  4967.2  1818.8
  4980.3 1807.91  4990.4 1805.53  5059.9 1804.35  5060.4 1803.85  5081.8 1804.35
    5110 1805.08    5141 1830.49    5161 1852.09    5171  1868.9    5181 1918.96
    5211 1935.73  5216.1 1940.94  5251.1 1953.98  5331.1 1976.02  5466.1 1985.46
#Mann= 8 ,-1 , 0
  4255.5     .07       0    4541    .035       0  4801.1     .07       0
  4814.9    .035       0  4967.2     .07       0  5059.9     .05       0
  5081.8     .07       0    5110      .1       0
Bank Sta=5059.9,5081.8
XS Rating Curve= 0 ,0
Exp/Cntr=0.3,0.1

Type RM Length L Ch R = 1 ,88464   ,585,585,585
BEGIN DESCRIPTION:
Turtle Creek 143.0
END DESCRIPTION:
XS GIS Cut Line= 3
      1890925.01     13904525.01        1891725.       13904825.
        1892125.       13904775.
#Sta/Elev= 30
  4155.7 1886.23  4250.9 1874.04  4341.7 1867.94  4427.1  1858.9  4452.1  1850.5
  4487.2  1843.2  4537.5 1833.52  4592.7 1828.13  4732.4 1822.05    4849    1823
  4884.6 1820.51  4916.3 1815.04    4946 1805.89  4956.7 1805.74    4967  1802.7
  4967.5  1802.2    4989  1802.7  5020.2 1803.71  5040.3 1806.88  5047.9 1814.35
  5052.9 1812.92  5060.5 1822.01  5090.7 1845.15  5100.8 1882.34  5110.9 1909.89
  5120.9 1917.08  5133.5 1920.76  5209.1 1953.04  5302.3  1975.9  5413.2 1986.77
#Mann= 5 ,-1 , 0
  4155.7     .07       0  4487.2    .035       0  4916.3     .07       0
    4967     .05       0    4989      .1       0
Bank Sta=4967,4989
XS Rating Curve= 0 ,0
Exp/Cntr=0.3,0.1

Type RM Length L Ch R = 1 ,87879   ,504,504,504
BEGIN DESCRIPTION:
Turtle Creek 142.0
END DESCRIPTION:
XS GIS Cut Line= 3
      1890974.99     13905625.01      1891653.36     13905315.92
      1891974.97     13905075.02
#Sta/Elev= 30
  4285.7 1913.27  4329.7 1909.25  4369.9 1895.15  4392.2 1876.91  4428.6 1855.48
  4450.6  1844.6  4489.9 1833.55  4582.1 1821.78  4687.5  1819.7  4857.6 1815.07
  4965.7 1804.13  4967.3 1803.72  4967.8 1803.22  4989.3 1803.72  5046.5 1805.71
  5054.8 1813.97  5061.1 1812.78  5069.4 1821.64  5075.7 1820.72  5090.3 1833.26
  5096.5 1831.55  5104.8 1839.21  5111.1 1835.82  5119.4 1841.51  5125.7 1838.48
  5140.3 1851.29  5146.5 1851.16  5154.9 1858.19  5311.1 1904.57    5433 1929.76
#Mann= 6 ,-1 , 0
  4285.7     .07       0  4369.9      .1       0  4687.5    .035       0
  4965.7      .1       0  4967.3     .05       0  4989.3      .1       0
Bank Sta=4967.3,4989.3
XS Rating Curve= 0 ,0
Exp/Cntr=0.3,0.1

Type RM Length L Ch R = 1 ,87375   ,476,476,476
BEGIN DESCRIPTION:
Turtle Creek 141.0
END DESCRIPTION:
XS GIS Cut Line= 3
      1891174.97     13905975.02        1891525.       13905775.
      1892324.98     13905125.01
#Sta/Elev= 30
  4592.9 1914.91    4644 1911.24  4665.6 1905.26  4673.6 1901.46  4681.5 1888.64
  4703.1 1868.06  4784.7 1827.47  4789.5 1823.92  4811.8 1823.63  4842.7 1817.81
  4938.5 1811.78    5013 1802.83  5013.5 1802.33    5035 1802.83  5085.6  1803.6
  5151.9 1805.77    5212 1815.82  5386.8 1838.59  5408.4 1839.41  5450.7 1848.01
  5485.9 1851.07  5589.9 1878.67  5621.7 1889.93  5714.4 1912.42  5756.2 1919.71
    5871 1953.73  5912.6 1960.86  5934.9 1970.46  6013.2 1991.81  6026.8 1992.97
#Mann= 7 ,-1 , 0
  4592.9      .1       0  4784.7     .07       0    5013     .05       0
    5035     .07       0  5085.6      .1       0    5212     .07       0
  5589.9      .1       0
Bank Sta=5013,5035
XS Rating Curve= 0 ,0
Exp/Cntr=0.3,0.1

Type RM Length L Ch R = 1 ,86899   ,656,656,656
BEGIN DESCRIPTION:
Turtle Creek 140.0
END DESCRIPTION:
XS GIS Cut Line= 4
      1891225.04       13906275.      1891499.28       13906275.
      1891728.71     13906177.77      1892424.97     13905525.03
#Sta/Elev= 30
  4534.5 1914.23  4714.5 1903.46  4724.5 1894.31  4734.5 1874.39  4804.1 1835.35
  4808.7 1835.35    4821 1822.71  4841.6 1809.95  4844.6 1807.83  4873.7 1806.88
    4891 1803.45  4933.7 1802.72  4934.2 1802.22  4955.8 1802.72  4988.7 1803.15
  5050.3 1812.93  5099.7 1815.95  5281.8 1815.96  5468.7  1818.1  5524.1 1824.57
  5587.6  1825.8  5609.1 1830.54  5644.3 1832.88  5672.6  1847.4  5679.9 1847.97
  5719.5 1867.12  5842.6 1916.38  5920.3 1930.24  5991.1 1948.87  6012.3 1956.56
#Mann= 7 ,-1 , 0
  4534.5      .1       0  4841.6     .07       0  4933.7     .05       0
  4955.8     .07       0  5281.8    .035       0  5468.7     .07       0
  5719.5      .1       0
Bank Sta=4933.7,4955.8
XS Rating Curve= 0 ,0
Exp/Cntr=0.3,0.1

Type RM Length L Ch R = 1 ,86243   ,534,534,534
BEGIN DESCRIPTION:
Turtle Creek 139.0
END DESCRIPTION:
XS GIS Cut Line= 3
      1891574.99     13907075.02        1891775.       13906725.
        1892575.       13905925.
#Sta/Elev= 30
  4603.2 1899.23  4670.2 1886.57    4735 1869.36  4772.4 1862.67  4778.1 1858.71
  4809.8 1852.96  4845.1 1849.38    4853 1846.89  4874.6 1830.43  4880.4 1823.89
  4902.7 1808.31  4939.4 1800.58    4972 1799.84  4972.5 1799.34  4994.6 1799.84
  5048.8 1800.79  5133.6 1806.87  5207.6 1808.36  5359.9 1813.24    5473 1814.57
  5627.2 1813.34  5827.1 1814.46  5883.1 1816.57  5911.4 1822.32    5937 1831.34
  5982.1 1854.22    6067 1906.33  6095.3 1921.78  6134.2 1939.24  6137.7 1939.24
#Mann= 7 ,-1 , 0
  4603.2     .07       0    4972     .05       0  4994.6     .07       0
  5207.6     .07       0  5627.2    .035       0  5827.1     .07       0
    5937      .1       0
Bank Sta=4972,4994.6
XS Rating Curve= 0 ,0
Exp/Cntr=0.3,0.1

Type RM Length L Ch R = 1 ,85709   ,652,652,652
BEGIN DESCRIPTION:
Turtle Creek 138.0
END DESCRIPTION:
XS GIS Cut Line= 3
      1891575.02     13907524.98        1892175.       13907025.
      1892725.04     13906774.98
#Sta/Elev= 30
  4219.5 1943.33  4356.8 1916.06  4432.3 1896.62  4460.9 1871.32  4510.4 1850.67
  4524.7 1848.52    4539 1839.88  4553.4 1836.78  4559.9 1841.07    4582 1832.13
  4602.8 1829.54  4617.1    1822  4654.5 1819.66  4709.6 1813.99  4880.1 1809.71
  4894.4 1808.34  4900.9 1803.24  4936.1 1799.96  5044.1 1799.95  5044.6 1799.45
  5066.7 1799.95  5251.7 1807.02  5400.3 1809.38  5451.9 1824.77  5501.9 1853.38
  5521.2 1862.97  5544.2  1883.5  5560.7 1892.36  5572.8 1914.06  5604.7 1918.49
#Mann= 8 ,-1 , 0
  4219.5     .07       0  4356.8      .1       0  4654.5     .07       0
  5044.1     .05       0  5066.7     .07       0  5251.7      .1       0
  5451.9     .07       0  5501.9      .1       0
Bank Sta=5044.1,5066.7
XS Rating Curve= 0 ,0
Exp/Cntr=0.3,0.1

Type RM Length L Ch R = 1 ,85057   ,276,276,276
BEGIN DESCRIPTION:
Turtle Creek 137.0
END DESCRIPTION:
XS GIS Cut Line= 5
      1891824.98     13908125.02      1892541.74     13907486.25
       1892597.3     13907422.02       1892678.9     13907390.77
      1892829.51     13907079.15
#Sta/Elev= 30
  3925.2 1935.48  4003.4 1912.25  4024.3 1898.35  4045.8 1874.51  4098.6 1840.96
  4123.8 1828.73  4173.1 1816.88  4248.2 1809.48  4401.4 1806.69    4743 1806.51
  4794.9 1806.22  4852.9 1805.72  4884.1 1794.25  4978.3 1793.26  4987.9 1792.79
  4988.4 1792.29  5010.5 1792.79  5029.2 1793.76  5034.6 1799.54  5042.7  1797.7
  5064.8 1806.75  5138.6 1808.01  5199.5 1810.41  5232.6 1818.73  5307.8 1852.13
  5319.5 1867.25  5330.4 1870.24  5358.6  1887.7  5364.1  1894.8  5403.7 1902.86
#Mann= 12 ,-1 , 0
  3925.2      .1       0  4098.6     .07       0  4248.2      .1       0
  4401.4     .07       0    4743    .035       0  4794.9     .07       0
  4978.3    .033       0  4987.9    .033       0  5010.5    .033       0
  5138.6      .1       0  5199.5     .07       0  5232.6      .1       0
Bank Sta=4987.9,5010.5
XS Rating Curve= 0 ,0
Exp/Cntr=0.3,0.1

Type RM Length L Ch R = 1 ,84781   ,766,766,766
BEGIN DESCRIPTION:
Mapping XS e0c6ea53
END DESCRIPTION:
XS GIS Cut Line= 3
       1892645.4     13908640.14      1892749.79     13907700.04
      1892848.14     13907089.69
#Sta/Elev= 30
  3929.8 1977.59  4005.4 1969.29  4061.4 1953.17  4116.1 1946.23  4281.7 1910.55
  4307.2 1906.74  4317.3 1878.55  4327.4 1863.34  4358.8 1845.58  4423.8    1814
  4478.3 1804.36  4548.6 1804.04  4554.9 1803.71    4580 1802.88  4653.5 1803.24
  4752.2 1803.73  4850.8 1787.13  4949.8 1787.18  4970.7 1786.94  4971.2 1786.44
  4993.4 1786.94  5032.7  1789.1  5048.9 1795.39  5093.5  1803.9  5174.5 1804.81
  5195.6 1810.79  5257.4 1809.37  5346.3 1852.04    5448 1895.07  5493.9 1900.52
#Mann= 14 ,-1 , 0
  3929.8      .1       0  4281.7     .07       0  4358.8      .1       0
  4548.6     .07       0  4554.9    .035       0    4580     .07       0
  4653.5    .035       0  4752.2     .07       0  4850.8      .1       0
  4949.8    .033       0  4970.7    .033       0  4993.4    .033       0
  5048.9     .07       0  5346.3      .1       0
Bank Sta=4970.7,4993.4
XS Rating Curve= 0 ,0
Exp/Cntr=0.3,0.1

Type RM Length L Ch R = 1 ,84015   ,482,482,482
BEGIN DESCRIPTION:
Turtle Creek 136.0
END DESCRIPTION:
XS GIS Cut Line= 3
      1893674.98     13908024.99        1893325.       13907825.
      1892874.98     13907024.97
#Sta/Elev= 30
  4597.9 1957.08  4620.9  1951.1  4627.4 1945.88  4847.7 1846.33  4862.8 1833.57
  4869.3 1818.15    4875 1809.55  4885.1 1803.53  4897.3 1791.57  4920.4 1780.03
  4944.2 1778.57  4944.7 1778.07    4967 1778.57  4992.6 1778.77  5046.6 1778.75
  5075.2 1793.88  5219.9 1801.14  5236.8 1801.17  5361.2 1801.63  5494.3 1806.02
    5538 1812.93  5587.1 1812.68    5619 1831.45  5671.1 1845.96  5705.6 1860.99
  5712.3 1867.11  5770.7  1875.2  5792.7 1884.28  5845.9 1898.79  5918.9 1908.03
#Mann= 9 ,-1 , 0
  4597.9      .1       0  4944.2    .033       0    4967      .1       0
  4992.6    .033       0  5075.2      .1       0  5219.9     .07       0
  5236.8      .1       0  5361.2    .035       0  5671.1      .1       0
Bank Sta=4944.2,4967
XS Rating Curve= 0 ,0
Exp/Cntr=0.3,0.1

Type RM Length L Ch R = 1 ,83533   ,577,577,577
BEGIN DESCRIPTION:
Turtle Creek 135.0
END DESCRIPTION:
XS GIS Cut Line= 3
      1893874.98     13907824.97      1893692.34     13907562.68
      1892925.03     13906975.02
#Sta/Elev= 30
    4607 1957.43  4635.3 1951.67  4751.4 1899.04  4843.9 1850.06  4850.7 1835.75
  4864.8 1822.07  4894.5 1808.24  4915.4 1791.35  4954.2 1778.67  4954.7 1778.17
    4977 1778.67  5057.3 1780.67  5094.4 1790.73  5149.5 1794.94  5305.4 1799.48
  5501.5 1810.53  5528.6 1820.73  5551.4 1823.11    5593 1835.55  5628.6 1838.05
  5651.1 1849.49  5671.9 1852.83  5680.9 1858.36    5701 1864.07  5707.3 1862.53
  5715.5  1867.6  5721.8 1866.29  5736.3 1874.58  5815.2 1897.02  5893.1 1906.56
#Mann= 7 ,-1 , 0
    4607      .1       0  4954.2     .05       0    4977      .1       0
  5057.3     .07       0  5149.5    .035       0  5305.4     .07       0
  5680.9      .1       0
Bank Sta=4954.2,4977
XS Rating Curve= 0 ,0
Exp/Cntr=0.3,0.1

Type RM Length L Ch R = 1 ,82956   ,596,596,596
BEGIN DESCRIPTION:
Turtle Creek 134.0
END DESCRIPTION:
XS GIS Cut Line= 3
      1894225.03     13907275.01        1893875.       13907075.
      1893124.99       13906725.
#Sta/Elev= 30
  4601.7 1931.13    4696 1916.33  4733.5 1902.17  4792.5 1868.55  4814.1 1860.15
  4851.5 1839.15  4910.5 1813.99  4932.1 1796.59  4953.7 1784.76  4979.7 1779.66
  4980.2 1779.16  5002.6 1779.66  5052.7 1780.36  5082.1 1780.38  5133.3 1789.59
  5159.9 1792.04  5350.1 1798.58  5441.5 1807.05  5479.4 1806.38    5486 1808.05
  5515.6 1814.13  5545.6 1825.01  5589.7 1833.71  5607.1 1846.67  5613.2 1846.94
  5652.8 1862.18  5681.1 1868.38  5772.6 1898.52  5797.5 1901.52  5832.5 1904.27
#Mann= 8 ,-1 , 0
  4601.7      .1       0  4979.7     .05       0  5002.6      .1       0
  5052.7     .07       0  5159.9    .035       0    5486     .07       0
  5613.2      .1       0  5797.5     .07       0
Bank Sta=4979.7,5002.6
XS Rating Curve= 0 ,0
Exp/Cntr=0.3,0.1

Type RM Length L Ch R = 1 ,82360   ,491,491,491
BEGIN DESCRIPTION:
Turtle Creek 133.0
END DESCRIPTION:
XS GIS Cut Line= 3
      1894374.97     13906824.98      1894091.59     13906598.08
      1893225.03     13906425.01
#Sta/Elev= 30
  4569.9 1918.37  4605.9 1914.23  4655.5 1901.31  4754.7 1854.93  4833.2 1823.49
  4839.6 1818.29  4847.6 1817.86    4854 1809.72    4862 1808.12  4868.4 1801.77
  4876.4 1799.02  4882.8 1802.43  4897.2 1785.94  4931.4 1779.92  4997.8  1779.6
  5009.2 1779.47  5009.7 1778.97  5032.1 1779.47  5173.7 1791.67  5272.1 1793.98
  5381.2 1796.27  5508.3 1807.81  5638.1 1838.15    5684 1855.72  5689.1 1855.38
    5735 1876.61  5740.1 1876.18  5755.4 1886.18    5786 1899.45  5816.6 1905.44
#Mann= 7 ,-1 , 0
  4569.9      .1       0  4997.8     .07       0  5009.2     .05       0
  5032.1     .07       0  5272.1    .035       0  5381.2     .07       0
  5508.3      .1       0
Bank Sta=5009.2,5032.1
XS Rating Curve= 0 ,0
Exp/Cntr=0.3,0.1

Type RM Length L Ch R = 1 ,81869   ,550,550,550
BEGIN DESCRIPTION:
Turtle Creek 132.0
END DESCRIPTION:
XS GIS Cut Line= 3
        1894475.       13906425.        1894075.       13906175.
        1893275.       13906175.
#Sta/Elev= 30
  4532.5 1908.34  4582.6 1898.42  4671.1    1862  4698.2 1846.89  4750.1 1832.29
  4765.4 1822.23  4771.3 1822.72  4786.6 1813.59  4807.9 1807.69  4815.5 1801.07
  4839.8 1788.43  4859.7 1777.88  4872.3 1775.08  4909.9 1769.22  4969.8 1768.87
  4970.3 1768.37  4992.7 1768.87  5001.2 1778.38  5022.2 1781.81  5044.2 1788.75
  5084.2 1792.35  5244.2 1792.32  5395.4 1796.31  5424.2 1798.37  5444.2 1803.31
  5474.2 1803.87  5654.2 1862.46  5754.2 1902.37  5774.2  1907.3  5804.2 1909.17
#Mann= 7 ,-1 , 0
  4532.5      .1       0  4839.8     .07       0  4872.3      .1       0
  4969.8     .05       0  4992.7      .1       0  5022.2    .035       0
  5395.4      .1       0
Bank Sta=4969.8,4992.7
XS Rating Curve= 0 ,0
Exp/Cntr=0.3,0.1

Type RM Length L Ch R = 1 ,81319   ,544,544,544
BEGIN DESCRIPTION:
Turtle Creek 131.0
END DESCRIPTION:
XS GIS Cut Line= 3
      1894675.02     13906175.02        1894225.       13905675.
      1893425.01       13905675.
#Sta/Elev= 30
  4327.4 1902.88  4369.7  1898.6  4532.6    1849  4615.8 1831.54  4638.7 1829.49
  4674.6 1817.17  4717.2  1813.4  4759.1 1798.79  4768.9 1797.83  4809.1 1796.59
  4823.3 1793.71  4830.1 1787.55  4837.5  1786.8  4844.3 1781.95  4899.6 1775.86
  4915.3 1775.69  4953.1  1767.6  4953.6  1767.1  4976.1  1767.6  5030.1 1768.04
  5113.2 1775.45  5150.1 1783.51  5200.1 1789.88  5290.1 1789.94  5403.9 1795.07
  5540.1  1808.6  5590.1 1818.05  5644.9 1833.11  5710.1 1852.07  5800.1 1886.29
#Mann= 9 ,-1 , 0
  4327.4      .1       0  4615.8     .07       0  4768.9      .1       0
  4899.6     .07       0  4953.1     .05       0  4976.1     .07       0
  5113.2    .035       0  5403.9     .07       0  5644.9      .1       0
Bank Sta=4953.1,4976.1
XS Rating Curve= 0 ,0
Exp/Cntr=0.3,0.1

Type RM Length L Ch R = 1 ,80775   ,547,547,547
BEGIN DESCRIPTION:
Turtle Creek 130.0
END DESCRIPTION:
XS GIS Cut Line= 3
      1894875.02     13905975.02        1894275.       13905175.
      1893925.01     13904725.01
#Sta/Elev= 30
  4000.1 1895.65  4092.8 1873.46    4172 1858.94  4200.1 1850.06  4236.6 1844.12
  4257.4 1837.74  4400.1 1820.19  4592.8 1802.49  4613.7 1795.14  4657.4  1797.9
  4700.1 1796.04    4722 1792.01  4750.1 1781.06  4757.4 1780.09    4880 1773.31
  4982.1 1768.31  5039.3 1762.26  5039.8 1761.76  5062.4 1762.26  5102.4 1764.12
  5121.4 1765.86  5127.7 1771.61  5135.9 1774.08  5141.9  1779.5  5156.7 1785.93
  5241.7 1790.61  5278.8  1803.6  5463.4 1909.23  5527.7 1936.91  5570.2 1949.62
#Mann= 7 ,-1 , 0
  4000.1      .1       0    4880     .07       0  4982.1      .1       0
  5039.3     .05       0  5062.4      .1       0  5102.4     .07       0
  5141.9      .1       0
Bank Sta=5039.3,5062.4
XS Rating Curve= 0 ,0
Exp/Cntr=0.3,0.1

Type RM Length L Ch R = 1 ,80228   ,550,550,550
BEGIN DESCRIPTION:
Turtle Creek 129.0
END DESCRIPTION:
XS GIS Cut Line= 3
      1894924.98     13905524.96        1894525.       13904725.
        1894175.       13904525.
#Sta/Elev= 30
  4105.4 1821.97  4180.8 1812.76  4225.5 1812.49  4259.9 1807.58  4418.4 1793.11
  4611.8  1784.9  4755.1 1782.34  4851.6 1778.73  4946.7 1763.58  4979.8  1761.9
  4980.3  1761.4  5002.9  1761.9  5022.8 1763.99  5045.1 1773.56  5050.9 1780.29
  5066.7 1788.08  5131.5 1835.42  5153.1 1860.01    5161 1877.92  5168.9 1881.82
  5174.7 1888.73  5190.5 1892.75  5196.3 1898.25  5206.4 1900.51  5255.3 1923.02
  5271.2 1924.39  5276.9 1928.34    5287 1929.03    5336 1944.78  5402.9 1953.07
#Mann= 6 ,-1 , 0
  4105.4     .07       0  4259.9      .1       0  4611.8     .07       0
  4755.1      .1       0  4979.8     .05       0  5002.9      .1       0
Bank Sta=4979.8,5002.9
XS Rating Curve= 0 ,0
Exp/Cntr=0.3,0.1

Type RM Length L Ch R = 1 ,79678   ,530,530,530
BEGIN DESCRIPTION:
Turtle Creek 128.0
END DESCRIPTION:
XS GIS Cut Line= 3
        1895125.     13905375.03        1895025.       13904575.
      1894725.02     13904275.02
#Sta/Elev= 30
  4193.6 1811.22  4195.1 1811.22  4236.5 1809.14  4284.3 1800.51  4317.1 1798.22
    4375 1786.44  4586.7 1780.85  4625.5 1781.15    4725 1781.16  4868.8 1780.52
  4876.4 1778.28  4881.4 1778.96    4889 1774.24  4919.2 1766.22  4929.3 1761.17
  4979.7 1761.78  5002.4  1758.9  5002.9  1758.4  5025.6  1758.9  5070.6 1769.77
  5098.9 1778.39  5127.1 1789.79    5212 1834.86  5226.1 1852.98  5240.3 1916.17
  5254.4 1919.03  5282.7 1920.66  5342.8 1920.53  5420.8 1918.32  5424.1 1918.32
#Mann= 8 ,-1 , 0
  4193.6     .07       0  4195.1      .1       0  4625.5    .035       0
    4725      .1       0  5002.4     .05       0  5025.6      .1       0
  5342.8     .07       0  5420.8      .1       0
Bank Sta=5002.4,5025.6
XS Rating Curve= 0 ,0
Exp/Cntr=0.3,0.1

Type RM Length L Ch R = 1 ,79148   ,526,526,526
BEGIN DESCRIPTION:
Turtle Creek 127.0
END DESCRIPTION:
XS GIS Cut Line= 3
      1895174.98     13905375.04        1895475.       13904725.
      1895424.99     13904324.95
#Sta/Elev= 30
  4283.9  1809.6    4361 1804.73    4367 1801.73  4418.4 1796.71  4458.8 1787.02
  4481.7 1783.98  4671.4 1778.87  4911.3 1777.17  4916.8 1776.97  4932.4 1769.41
  4955.8 1760.38  4985.5 1756.89    4986 1756.39  5008.7 1756.89  5042.7 1758.79
  5100.6 1771.21  5118.3 1778.92  5123.3 1777.39  5198.9 1832.04  5203.9 1829.53
  5231.6 1853.01  5251.8 1865.84  5261.9 1875.23  5271.9 1903.82  5279.5  1908.5
  5284.5 1907.91  5312.2  1913.3  5342.5  1913.1  5365.2  1911.5    5403 1905.31
#Mann= 5 ,-1 , 0
  4283.9      .1       0  4671.4    .035       0  4932.4      .1       0
  4985.5     .05       0  5008.7      .1       0
Bank Sta=4985.5,5008.7
XS Rating Curve= 0 ,0
Exp/Cntr=0.3,0.1

Type RM Length L Ch R = 1 ,78622   ,537,537,537
BEGIN DESCRIPTION:
Turtle Creek 126.0
END DESCRIPTION:
XS GIS Cut Line= 3
      1895125.02     13905724.98        1895925.       13904925.
      1896275.04     13904724.98
#Sta/Elev= 30
  3863.4 1839.02  3905.8 1832.23  3962.4 1818.56  3990.7 1818.74  4149.4 1804.68
  4273.5 1797.71  4372.5  1784.4  4544.9 1779.95  4810.9 1775.62  4839.2 1774.59
    4878    1769  4980.6 1759.25  4991.1 1755.37  4991.6 1754.87  5014.3 1755.37
  5061.7 1760.31  5104.9 1776.29  5110.6 1782.16  5122.7  1787.8    5133 1797.23
  5142.3 1800.55  5148.1 1807.42  5163.2 1814.38    5179 1824.98  5191.3 1839.23
  5201.3 1847.34  5232.9 1879.66  5250.3 1891.31  5330.9  1915.4  5397.9 1919.87
#Mann= 9 ,-1 , 0
  3863.4     .07       0  4149.4      .1       0  4544.9    .035       0
    4878     .07       0  4991.1     .05       0  5014.3     .07       0
  5122.7    .033       0  5163.2     .07       0  5232.9      .1       0
Bank Sta=4991.1,5014.3
XS Rating Curve= 0 ,0
Exp/Cntr=0.3,0.1

Type RM Length L Ch R = 1 ,78085   ,544,544,544
BEGIN DESCRIPTION:
Turtle Creek 125.0
END DESCRIPTION:
XS GIS Cut Line= 3
        1896375.     13905974.99        1896375.       13905175.
        1896375.     13904774.99
#Sta/Elev= 30
  4200.2 1816.07  4250.2 1809.75  4280.2 1799.63  4290.2 1800.48  4330.2 1783.66
  4360.2 1776.46  4420.2 1770.99  4498.5 1769.85  4550.2 1767.62  4596.8 1768.85
  4680.5 1766.37  4720.2 1765.07  4760.2 1772.01  4780.2 1772.97  4960.2 1763.54
  4997.7 1755.92    5042 1756.05  5048.6 1755.86  5049.1 1755.36  5071.8 1755.86
  5110.2 1764.77  5130.2 1776.59  5140.2 1783.26  5160.2 1801.74  5220.2 1839.37
  5250.2 1874.16  5270.2 1889.85  5300.2 1907.98  5330.2 1918.71  5400.2 1922.14
#Mann= 7 ,-1 , 0
  4200.2      .1       0  4498.5     .07       0  4596.8      .1       0
  4680.5     .07       0    5042      .1       0  5048.6     .05       0
  5071.8      .1       0
Bank Sta=5048.6,5071.8
XS Rating Curve= 0 ,0
Exp/Cntr=0.3,0.1

Type RM Length L Ch R = 1 ,77541   ,136,136,136
BEGIN DESCRIPTION:
Turtle Creek 124.0
END DESCRIPTION:
XS GIS Cut Line= 3
      1896675.01     13906174.97        1896825.       13905375.
        1896775.     13904975.02
#Sta/Elev= 30
  4190.4 1841.79  4272.1  1826.7  4363.3 1808.75  4437.1 1800.05  4475.2 1784.88
  4507.4 1780.06  4542.2  1772.4  4627.9 1760.82  4668.6 1762.87  4710.1 1769.11
  4729.6 1766.97  4739.8  1763.1  4784.1 1761.85  4891.2 1760.07  4943.3 1755.12
  4978.4 1757.04  4990.2 1754.75  4990.7 1754.25  5013.4 1754.75  5105.1 1757.19
  5127.8 1761.39  5145.4  1770.5  5175.6  1778.3  5203.3  1790.1  5208.4 1789.89
    5284 1835.45    5289 1835.98  5296.6 1842.28  5364.6 1880.03  5407.4  1899.6
#Mann= 8 ,-1 , 0
  4190.4      .1       0  4272.1     .07       0  4507.4      .1       0
  4784.1     .07       0  4891.2      .1       0  4978.4     .07       0
  4990.2     .05       0  5013.4      .1       0
Bank Sta=4990.2,5013.4
XS Rating Curve= 0 ,0
Exp/Cntr=0.3,0.1

Type RM Length L Ch R = 1 ,77405   ,443,443,443
BEGIN DESCRIPTION:
Mapping XS c488dab6
END DESCRIPTION:
XS GIS Cut Line= 3
      1897074.17     13906270.52      1896935.27     13905426.74
      1896814.02     13904959.04
#Sta/Elev= 30
  4093.6 1851.27  4129.6 1839.93  4190.4  1826.3  4329.9 1807.29  4433.6 1796.37
  4443.8  1792.7    4489 1790.87  4550.2 1783.38  4717.4 1770.47    4875 1764.43
  4926.5 1762.15  4947.1 1757.46  4977.1 1755.37  4989.1 1754.94  4989.6 1754.44
  5015.2 1754.94  5089.6 1757.27  5136.5 1773.01  5211.4 1791.87  5239.8 1804.63
  5246.8 1810.23    5252 1809.87  5281.1 1824.14  5322.4 1846.71    5328 1852.39
  5368.6 1870.73  5374.1 1877.12    5404 1894.28  5409.2 1894.56  5431.9  1905.5
#Mann= 7 ,-1 , 0
  4093.6      .1       0  4329.9     .07       0    4875      .1       0
  4926.5     .07       0  4977.1      .1       0  4989.1     .05       0
  5015.2      .1       0
Bank Sta=4989.1,5015.2
XS Rating Curve= 0 ,0
Exp/Cntr=0.3,0.1

Type RM Length L Ch R = 1 ,76962   ,546,546,546
BEGIN DESCRIPTION:
Turtle Creek 123.0
END DESCRIPTION:
XS GIS Cut Line= 3
      1897925.03     13906325.04        1897275.       13905525.
      1896975.02     13904925.04
#Sta/Elev= 30
  3963.2 1922.65  4027.7 1908.32  4055.2 1898.27    4127 1860.24  4147.8 1854.29
  4176.6 1840.12  4240.5 1815.73  4283.6 1804.41  4446.7 1785.32  4481.9    1787
  4615.3 1778.68  4625.1 1778.69  4716.4  1773.7  4916.5 1763.87  4937.3 1759.41
  4972.5 1762.14  5002.4 1756.68  5106.8 1754.98  5107.3 1754.48  5132.9 1754.98
  5209.2 1762.06  5270.7 1773.28    5321 1775.31  5343.4 1779.14  5360.2 1786.16
  5365.8 1784.91  5499.9 1834.61  5539.1 1855.91  5606.1 1886.24  5664.8 1901.87
#Mann= 6 ,-1 , 0
  3963.2      .1       0  4615.3     .07       0  4625.1    .063       0
  4716.4      .1       0  5106.8     .05       0  5132.9      .1       0
Bank Sta=5106.8,5132.9
XS Rating Curve= 0 ,0
Exp/Cntr=0.3,0.1

Type RM Length L Ch R = 1 ,76416   ,525,525,525
BEGIN DESCRIPTION:
Turtle Creek 122.0
END DESCRIPTION:
XS GIS Cut Line= 3
      1898125.01     13906175.02      1897746.69       13905498.
      1897124.97     13904824.97
#Sta/Elev= 30
  4228.3 1915.22  4251.2 1913.35  4279.6 1906.38  4317.4    1883  4388.7 1847.27
  4469.3  1812.9    4523 1795.23  4566.4 1782.33  4617.8 1779.76  4674.6  1771.9
    4859 1764.75  4918.2 1761.71  4955.9  1749.6  4973.7 1750.25  5015.3 1749.32
  5015.8 1748.82  5041.5 1749.32  5085.1 1755.06  5194.1 1760.17  5353.9 1771.84
  5438.9 1796.83  5544.9 1811.58  5545.2 1811.64  5665.2 1819.31  5686.7 1827.54
  5721.9 1835.52  5778.6 1860.63  5835.3 1874.03  5884.6 1889.64  5920.1 1893.45
#Mann= 9 ,-1 , 0
  4228.3      .1       0  4674.6    .035       0    4859     .07       0
  4973.7      .1       0  5015.3     .05       0  5041.5      .1       0
  5194.1      .1       0  5544.9     .07       0  5545.2      .1       0
Bank Sta=5015.3,5041.5
XS Rating Curve= 0 ,0
Exp/Cntr=0.3,0.1

Type RM Length L Ch R = 1 ,75891   ,544,544,544
BEGIN DESCRIPTION:
Turtle Creek 121.0
END DESCRIPTION:
XS GIS Cut Line= 3
        1898275.     13906124.97        1898225.       13905425.
      1897424.99     13904874.99
#Sta/Elev= 30
  4292.6 1913.51  4342.7 1906.78  4360.2 1896.24    4453  1851.5  4483.1 1839.67
  4523.2 1819.56  4583.3 1795.18  4623.4 1782.94  4633.4 1777.85    4667 1776.14
  4786.3 1768.52  4914.2 1764.99  4926.7 1762.38  4934.2 1755.67  4944.2 1750.45
  4966.9 1750.67  4978.8 1750.11  4979.3 1749.61    5005 1750.11  5173.2 1754.45
  5223.2 1757.68  5350.1 1763.53  5512.6 1771.81  5543.3 1775.39  5598.6 1779.79
    5677 1791.21  5721.6 1792.19  5818.3 1804.72    5886 1810.94  5965.2 1821.93
#Mann= 11 ,-1 , 0
  4292.6      .1       0    4667    .035       0  4966.9      .1       0
  4978.8     .05       0    5005      .1       0  5173.2     .07       0
  5223.2    .035       0  5350.1     .07       0  5543.3      .1       0
  5598.6    .035       0  5818.3     .07       0
Bank Sta=4978.8,5005
XS Rating Curve= 0 ,0
Exp/Cntr=0.3,0.1

Type RM Length L Ch R = 1 ,75347   ,530,530,530
BEGIN DESCRIPTION:
Turtle Creek 120.0
END DESCRIPTION:
XS GIS Cut Line= 3
      1899125.02       13905175.        1898625.       13905125.
      1897824.96     13904874.99
#Sta/Elev= 30
  4497.5 1921.81  4550.3 1911.16  4638.2 1857.11  4645.8 1850.82  4650.8 1851.09
  4658.3 1844.86  4746.3 1795.06  4751.3 1794.77  4758.8 1790.07    4789 1778.98
  4839.2 1770.85  4851.8 1765.76  4859.3 1758.16  4876.2 1747.63  4876.7 1747.13
  4902.7 1747.63  4939.7 1749.34  4979.9 1748.73  4997.5 1750.26  5040.8 1749.55
  5081.2 1750.02  5118.9 1754.06  5157.2 1756.01  5399.4  1761.2  5511.3 1763.28
  5519.1 1764.52    5550 1764.66  5609.8  1773.5  5784.2 1781.96  5838.2 1786.94
#Mann= 7 ,-1 , 0
  4497.5      .1       0  4876.2     .05       0  4902.7      .1       0
  5040.8     .07       0  5399.4    .035       0  5511.3     .07       0
  5609.8      .1       0
Bank Sta=4876.2,4902.7
XS Rating Curve= 0 ,0
Exp/Cntr=0.3,0.1

Type RM Length L Ch R = 1 ,74817   ,566,566,566
BEGIN DESCRIPTION:
Turtle Creek 119.0
END DESCRIPTION:
XS GIS Cut Line= 3
      1899124.99     13905074.99        1898875.       13904725.
      1898074.96       13904775.
#Sta/Elev= 30
  4565.2 1915.73  4622.9 1911.33  4657.4 1901.19  4664.7 1895.44  4673.3 1894.07
  4679.5 1887.18  4688.1 1886.21  4729.9 1865.68  4744.6  1862.6  4765.5 1849.65
  4845.4 1815.33  4851.5 1807.68  4860.1 1806.15  4872.4 1794.51    4881 1791.73
  4887.2 1781.53  4895.8 1780.65  4901.9  1772.8  4916.7 1769.75  4922.8  1762.2
  4931.4 1761.23  4937.5 1755.12    4967 1748.48  5052.1 1747.65  5052.6 1747.15
  5078.7 1747.65  5098.2 1749.73  5635.5 1762.25  5719.2 1764.84  5796.9 1774.05
#Mann= 5 ,-1 , 0
  4565.2      .1       0  5052.1     .05       0  5078.7      .1       0
  5098.2     .07       0  5635.5      .1       0
Bank Sta=5052.1,5078.7
XS Rating Curve= 0 ,0
Exp/Cntr=0.3,0.1

Type RM Length L Ch R = 1 ,74251   ,571,571,571
BEGIN DESCRIPTION:
Turtle Creek 118.0
END DESCRIPTION:
XS GIS Cut Line= 3
      1899225.03       13904275.        1898725.       13904275.
      1897924.98     13904525.01
#Sta/Elev= 30
  4504.5  1914.9  4524.5 1912.98  4534.5 1909.71  4684.5 1843.85  4764.5 1811.92
  4774.5 1807.34  4784.5 1790.58  4794.5 1783.98  4814.5 1779.24  4854.5 1759.37
  4874.5 1747.16  4904.5  1741.4  4931.2 1739.19  4931.7 1738.69  4957.8 1739.19
  4964.5 1742.19  4978.7 1740.65  5007.1 1740.79  5020.8 1746.17    5036 1747.53
  5085.7 1746.73  5124.7    1750    5358 1756.56  5426.2 1758.09  5453.5 1762.73
  5588.6 1762.69    5607 1764.33  5723.3 1773.56  5787.2  1779.7  5842.7 1783.92
#Mann= 9 ,-1 , 0
  4504.5      .1       0  4931.2    .035       0  4957.8      .1       0
  4978.7    .035       0  5124.7     .07       0    5358    .035       0
    5607      .1       0  5723.3     .07       0  5787.2      .1       0
Bank Sta=4931.2,4957.8
XS Rating Curve= 0 ,0
Exp/Cntr=0.3,0.1

Type RM Length L Ch R = 1 ,73680   ,301,301,301
BEGIN DESCRIPTION:
Turtle Creek 117.0
END DESCRIPTION:
XS GIS Cut Line= 3
      1898774.99     13903475.02        1898575.       13903825.
      1897774.97     13904475.02
#Sta/Elev= 30
  4596.9 1941.15  4642.2 1936.91  4677.5  1927.9    4707 1916.93  4744.4 1898.01
  4825.1 1849.98  4868.3 1819.64  4911.4 1793.28  4954.6 1770.58  4964.7 1767.33
  4970.5 1760.96  4983.8 1739.33  4984.3 1738.83  5010.5 1739.33  5049.6 1741.11
  5071.1 1740.86  5099.8 1744.89  5178.1 1744.25    5231 1747.44  5269.9 1754.63
  5381.1 1756.13  5582.5 1759.58  5654.4 1762.98    5672 1765.95  5732.7 1767.06
  5831.8 1780.56  5881.3 1783.54  5895.7  1787.4  5935.4 1788.74  6030.8 1794.89
#Mann= 9 ,-1 , 0
  4596.9      .1       0  4983.8     .05       0  5010.5      .1       0
  5049.6     .07       0    5231    .035       0  5269.9     .07       0
  5381.1    .035       0    5672     .07       0  5935.4      .1       0
Bank Sta=4983.8,5010.5
XS Rating Curve= 0 ,0
Exp/Cntr=0.3,0.1

Type RM Length L Ch R = 1 ,73379   ,259,259,259
BEGIN DESCRIPTION:
Turtle Creek 116.1
END DESCRIPTION:
XS GIS Cut Line= 4
      1898838.76     13903251.18      1898390.83     13903597.55
      1898289.27     13903667.86      1897573.12     13904222.55
#Sta/Elev= 30
  4438.8 1940.19  4671.6 1941.28  4708.7  1936.7    4744  1927.7  4822.8  1896.5
  4829.2  1877.1  4835.5 1865.24  4893.5 1821.14  4928.8 1788.88  4972.2 1759.95
  5003.7 1746.18  5022.6 1739.61  5064.4 1738.95    5066 1736.14  5066.5 1735.64
  5092.7 1736.14  5115.1 1740.16  5128.1 1736.17  5165.1 1744.41  5179.6 1752.07
  5227.9 1755.04  5349.8 1753.58  5527.5 1757.06  5571.6 1759.13  5685.7 1762.48
  5747.6 1771.04  5842.3 1786.73  5949.2 1791.19  6029.9 1801.32  6034.4  1801.4
#Mann= 9 ,-1 , 0
  4438.8      .1       0  5003.7     .07       0    5066     .05       0
  5092.7     .07       0  5227.9    .035       0  5527.5      .1       0
  5571.6    .035       0  5747.6     .07       0  6029.9      .1       0
Bank Sta=5066,5092.7
XS Rating Curve= 0 ,0
Exp/Cntr=0.3,0.1
