HEC-RAS study Turtle Creek.prj: Turtle Creek Base Level Engineering

--- Turtle Creek.g01 (geometry) --- (continued)

Type RM Length L Ch R = 1 ,73120   ,586,586,586
BEGIN DESCRIPTION:
Turtle Creek 116.0
END DESCRIPTION:
XS GIS Cut Line= 3
      1898524.96     13903275.02        1898175.       13903475.
      1897424.99     13904175.01
#Sta/Elev= 30
  4596.7 1928.77  4669.4 1927.72  4722.6 1915.99  4728.4 1871.74  4734.9 1864.64
  4803.3 1827.24  4815.5  1817.2  4830.6 1812.19  4861.6 1788.89  4896.1 1751.99
  4911.2 1743.75  4970.3 1732.22  5007.7 1731.13  5008.2 1730.63  5034.4 1731.13
  5056.2 1734.29  5077.7 1744.79  5112.9 1752.47  5274.1 1751.84  5413.4 1755.49
  5541.6 1757.83  5643.4 1759.76  5693.2 1764.37  5793.2 1787.56  5855.9 1790.11
  5862.8  1793.4  5912.6    1797  5958.5 1805.66  5967.5 1808.13  6025.7 1809.17
#Mann= 9 ,-1 , 0
  4596.7      .1       0  5007.7     .05       0  5034.4      .1       0
  5274.1    .035       0  5413.4      .1       0  5541.6    .035       0
  5793.2     .07       0  5958.5      .1       0  5967.5    .035       0
Bank Sta=5007.7,5034.4
XS Rating Curve= 0 ,0
Exp/Cntr=0.3,0.1

Type RM Length L Ch R = 1 ,72534   ,532,532,532
BEGIN DESCRIPTION:
Turtle Creek 115.0
END DESCRIPTION:
XS GIS Cut Line= 3
      1898374.95       13903025.        1897775.       13903075.
      1897075.03     13903824.97
#Sta/Elev= 30
    4393 1870.01  4450.6 1855.86  4455.7  1859.6  4473.2 1855.24  4571.1 1815.54
  4576.1 1816.66  4623.7 1800.67  4774.3 1770.89  4834.5 1748.57  4966.2 1730.89
  4979.1 1729.75  4979.6 1729.25  5005.9 1729.75    5009  1732.3  5044.6 1735.75
  5101.2 1737.07  5136.5 1743.44  5250.8 1749.13  5414.7 1754.03  5425.7 1754.28
  5635.8 1758.45  5699.6  1760.5  5794.5 1764.17  5865.7  1769.9  5886.4 1769.99
  5893.7 1772.95  5900.5  1781.2  5936.2 1788.71  5975.3 1792.12  6020.9 1795.41
#Mann= 12 ,-1 , 0
    4393      .1       0  4966.2    .035       0  4979.1    .035       0
  5005.9    .035       0  5101.2     .07       0  5250.8      .1       0
  5414.7     .07       0  5425.7      .1       0  5635.8     .07       0
  5699.6    .035       0  5865.7      .1       0  5975.3     .07       0
Bank Sta=4979.1,5005.9
XS Rating Curve= 0 ,0
Exp/Cntr=0.3,0.1

Type RM Length L Ch R = 1 ,72002   ,547,547,547
BEGIN DESCRIPTION:
Turtle Creek 114.0
END DESCRIPTION:
XS GIS Cut Line= 3
      1897925.03     13902274.97        1897325.       13902825.
      1897025.03     13903124.97
#Sta/Elev= 30
  4190.9 1792.76  4240.6 1790.87  4275.7 1784.92  4299.7 1777.96  4353.7 1770.02
  4381.8 1763.32    4396 1763.22  4427.1 1760.25  4523.6 1756.02  4615.5 1753.47
  4700.6 1749.15  4757.3 1747.94  4764.1    1745  4785.7 1742.73    4814 1737.08
  4892.9 1732.94  4948.5 1731.05  4962.6 1729.38  4969.4 1727.04  4970.1 1725.48
  4970.6 1724.98  4997.1 1725.48  5008.4 1725.71    5019 1733.77  5033.2 1738.37
  5051.4 1741.38  5089.7  1743.3  5181.7 1750.41  5310.7 1753.06  5429.1 1755.92
#Mann= 8 ,-1 , 0
  4190.9      .1       0  4299.7    .035       0  4427.1     .07       0
  4892.9      .1       0  4970.1     .05       0  4997.1      .1       0
  5051.4     .07       0  5310.7      .1       0
Bank Sta=4970.1,4997.1
XS Rating Curve= 0 ,0
Exp/Cntr=0.3,0.1

Type RM Length L Ch R = 1 ,71455   ,582,582,582
BEGIN DESCRIPTION:
Turtle Creek 113.0
END DESCRIPTION:
XS GIS Cut Line= 3
      1897774.96     13902175.01        1897075.       13902375.
      1896275.03     13903174.97
#Sta/Elev= 30
  4270.9 1791.26  4316.7 1788.98  4360.6 1773.28  4399.6 1767.17  4433.4 1755.21
    4513 1747.62  4698.4 1743.85  4831.3 1738.91  4884.5 1728.48  4963.2 1721.87
  4963.7 1721.37  4990.3 1721.87    5013 1732.54  5055.4 1740.58  5207.5 1747.86
  5232.3 1748.25  5485.7 1751.62  5510.2 1752.05  5629.7 1755.21    5645 1755.92
  5720.1 1760.17  5748.4 1769.09  5773.7 1766.61  5779.8 1766.25  5914.6  1780.8
  5960.5 1794.82  6031.2 1797.48  6073.7 1811.56  6110.8 1816.46  6130.2 1818.61
#Mann= 17 ,-1 , 0
  4270.9      .1       0  4316.7    .035       0    4513     .07       0
  4698.4      .1       0  4831.3     .07       0  4963.2     .05       0
  4990.3     .07       0  5207.5    .035       0  5232.3     .07       0
  5485.7    .035       0  5510.2     .07       0  5629.7    .035       0
    5645     .07       0  5773.7    .035       0  5779.8     .07       0
  5914.6    .035       0  6110.8     .07       0
Bank Sta=4963.2,4990.3
XS Rating Curve= 0 ,0
Exp/Cntr=0.3,0.1

Type RM Length L Ch R = 1 ,70873   ,566,566,566
BEGIN DESCRIPTION:
Turtle Creek 112.0
END DESCRIPTION:
XS GIS Cut Line= 3
      1897824.96     13902074.98        1897175.       13901825.
      1896875.03     13901525.03
#Sta/Elev= 30
  4307.9 1793.31  4352.9  1792.9  4367.4 1789.59  4402.1 1775.07  4425.7 1768.41
  4447.1 1759.51  4468.6 1752.98  4486.8 1748.53  4513.2  1746.4  4580.9 1743.14
    4790  1742.1  4810.8 1740.25  4843.6 1738.69  4874.6 1732.76  4918.6 1727.09
  4957.7 1725.37  4964.6 1724.69  4972.1 1720.75    4981 1720.72  4981.5 1720.22
  5008.2 1720.72  5032.6 1723.82  5060.8 1733.19  5117.4 1739.02  5231.8    1739
  5280.6 1737.83  5301.3 1739.53  5357.8 1754.29    5372 1756.61  5428.5 1758.54
#Mann= 10 ,-1 , 0
  4307.9      .1       0  4367.4    .035       0  4513.2     .07       0
  4580.9    .035       0  4810.8     .07       0  4957.7      .1       0
    4981     .05       0  5008.2      .1       0  5231.8    .035       0
  5280.6      .1       0
Bank Sta=4981,5008.2
XS Rating Curve= 0 ,0
Exp/Cntr=0.3,0.1

Type RM Length L Ch R = 1 ,70307   ,1077,1077,1077
BEGIN DESCRIPTION:
Turtle Creek 111.0
END DESCRIPTION:
XS GIS Cut Line= 3
      1897875.03     13902025.04        1897325.       13901375.
      1896584.24     13901313.83
#Sta/Elev= 30
  4143.9 1793.97  4186.2  1794.2  4200.5 1792.18  4222.5 1784.17  4235.6 1777.71
  4256.6 1771.31  4307.1 1753.07  4327.9 1748.54  4370.8 1743.69  4456.6 1740.33
  4619.1 1738.75  4789.9 1735.06  4803.7 1732.78  4832.3 1732.04    4896 1726.83
  4938.9 1725.94  4981.7 1723.07  4991.8 1719.74  4992.3 1719.24  5019.1 1719.74
  5053.7 1721.83  5065.7 1723.62  5075.7 1727.38  5095.8 1739.86  5105.8 1742.71
  5152.3 1744.82    5251 1744.37  5349.6 1745.04  5542.2  1747.3  5738.7 1755.36
#Mann= 9 ,-1 , 0
  4143.9      .1       0  4256.6    .035       0  4789.9     .07       0
  4991.8     .05       0  5019.1     .07       0  5053.7    .035       0
  5152.3     .07       0    5251    .035       0  5349.6     .07       0
Bank Sta=4991.8,5019.1
XS Rating Curve= 0 ,0
Exp/Cntr=0.3,0.1

Type RM Length L Ch R = 1 ,69230   ,630,630,630
BEGIN DESCRIPTION:
Turtle Creek 110.0
END DESCRIPTION:
XS GIS Cut Line= 4
        1898225.     13901574.99      1898071.85     13901126.18
        1898008.     13900891.81      1897769.36     13900203.33
#Sta/Elev= 30
  4532.5 1763.52  4579.5 1762.58  4594.1 1758.41  4610.8 1753.45    4617 1749.66
  4648.7 1738.32  4673.5  1735.1    4691  1734.9  4730.9 1729.69  4793.5 1725.27
  4902.3 1721.94  4918.8 1717.77  4978.3 1717.17  4979.3 1716.67  5016.5 1717.17
  5028.7 1717.61    5039 1720.22    5048 1727.21  5053.2 1726.22  5059.8  1733.3
  5070.1 1737.22  5101.2 1739.24  5128.9 1739.34  5231.7 1740.66    5398 1743.33
  5542.6  1747.4  5754.3 1754.57  5819.1 1758.05  5916.8 1766.73  5978.3 1774.63
#Mann= 7 ,-1 , 0
  4532.5    .035       0  4594.1      .1       0  4978.3     .05       0
  5016.5      .1       0  5128.9     .07       0  5231.7    .035       0
  5819.1      .1       0
Bank Sta=4978.3,5016.5
XS Rating Curve= 0 ,0
Exp/Cntr=0.3,0.1

Type RM Length L Ch R = 1 ,68600   ,528,528,528
BEGIN DESCRIPTION:
Turtle Creek 109.0
END DESCRIPTION:
XS GIS Cut Line= 4
      1898575.01     13901674.96        1898625.       13901275.
      1898613.83     13901089.87      1897933.49     13900219.82
#Sta/Elev= 30
  4592.2 1777.24  4594.6 1777.24  4715.6 1772.37  4773.6 1766.13  4783.6 1762.52
  4788.2 1758.27  4791.2 1755.49  4796.2 1755.86    4834 1729.47  4849.2 1722.74
    4948 1720.56  5036.3 1717.58  5037.3 1717.08  5074.5 1717.58  5095.5  1720.7
  5190.1 1726.96  5212.3 1730.56    5263 1732.15  5422.6 1735.41  5548.7 1737.32
  5584.4 1737.61  5846.6 1740.84  6129.8 1751.55    6145 1751.08  6194.8  1755.7
  6252.6 1765.18    6259 1764.38  6273.5 1768.84  6279.8 1768.47  6285.2 1771.35
#Mann= 12 ,-1 , 0
  4592.2      .1       0  4594.6     .07       0  4788.2      .1       0
  4849.2     .07       0    4948    .035       0  5036.3    .035       0
  5074.5    .035       0    5263     .07       0  5422.6    .035       0
  5548.7     .07       0  5584.4    .035       0  6129.8      .1       0
Bank Sta=5036.3,5074.5
XS Rating Curve= 0 ,0
Exp/Cntr=0.3,0.1

Type RM Length L Ch R = 1 ,68072   ,633,633,633
BEGIN DESCRIPTION:
Turtle Creek 108.0
END DESCRIPTION:
XS GIS Cut Line= 3
        1899025.     13901574.99        1899075.       13901175.
      1898133.35     13900090.58
#Sta/Elev= 30
  4591.9 1768.71  4853.9 1751.83    4864 1746.41  4871.5 1737.01  4876.6 1738.13
  4894.2 1719.24  5025.7  1716.7  5026.7  1716.2    5064  1716.7  5065.7 1719.72
    5080 1721.21    5177  1723.6  5264.2 1729.76  5306.9 1726.39  5430.3 1730.51
  5582.7 1734.07  5696.5 1735.75  5987.8 1738.87  6058.1 1741.97  6105.6 1748.85
  6164.4 1754.95  6192.9 1761.89  6207.2 1772.16  6299.3  1813.7  6313.5 1823.67
  6362.9 1836.79  6370.5  1841.7  6391.4 1844.03  6405.6 1852.82  6431.2 1854.11
#Mann= 8 ,-1 , 0
  4591.9      .1       0  5025.7     .05       0    5064     .07       0
    5177     .07       0  5430.3    .035       0  5582.7     .07       0
  5696.5    .035       0  6105.6      .1       0
Bank Sta=5025.7,5064
XS Rating Curve= 0 ,0
Exp/Cntr=0.3,0.1

Type RM Length L Ch R = 1 ,67439   ,529,529,529
BEGIN DESCRIPTION:
Turtle Creek 107.0
END DESCRIPTION:
XS GIS Cut Line= 4
      1899769.41     13901433.73      1899595.62     13900821.87
       1899354.3     13900589.23      1898874.98     13899924.97
#Sta/Elev= 30
  4174.6 1764.93  4815.9 1741.56  4823.1 1738.65    4839 1718.78  4858.4  1708.8
  4924.1 1707.37  4925.1 1706.87  4962.5 1707.37  4964.4 1716.67  5064.9 1718.52
  5105.8 1716.35  5134.1 1723.18  5204.5 1723.96    5327 1724.89    5392 1730.44
  5628.8 1735.28  5670.5 1740.97  5696.8 1751.52  5771.1 1786.08  5800.5 1806.25
  5821.4 1814.48  5836.1 1827.85  5842.3 1827.34  5850.8 1834.45    5857 1834.26
  5865.6  1841.4  5871.7 1842.52  5886.4  1858.8  5901.1 1868.27    5965 1900.93
#Mann= 7 ,-1 , 0
  4174.6     .07       0    4839    .033       0  4924.1    .033       0
  4962.5    .033       0  5064.9     .07       0  5204.5    .035       0
  5696.8      .1       0
Bank Sta=4924.1,4962.5
XS Rating Curve= 0 ,0
Exp/Cntr=0.3,0.1

Type RM Length L Ch R = 1 ,66910   ,560,560,560
BEGIN DESCRIPTION:
Turtle Creek 106.0
END DESCRIPTION:
XS GIS Cut Line= 3
      1899916.98     13901391.11        1899825.       13900425.
      1899024.99     13899824.99
#Sta/Elev= 30
    4025 1764.48  4308.5 1751.74  4493.2 1747.73  4730.5 1732.47  4864.9 1731.82
    4885 1728.48  4935.2    1711  4975.4 1708.33  4983.6 1704.74  4984.6 1704.24
    5022 1704.74  5067.4 1707.58  5102.8 1705.78  5123.6  1712.3  5202.8 1719.02
  5421.9 1722.47  5554.3 1731.13  5652.8 1741.78  5667.4 1745.41  5688.2 1756.68
    5709 1753.97  5731.9 1756.76    5759 1771.22  5838.2 1799.27  5902.8 1830.58
  5938.2 1842.47  5952.8 1850.63  5973.6 1856.08  5981.9 1862.06  5995.5 1866.58
#Mann= 5 ,-1 , 0
    4025     .07       0  4983.6     .05       0    5022     .07       0
  5421.9    .035       0  5554.3      .1       0
Bank Sta=4983.6,5022
XS Rating Curve= 0 ,0
Exp/Cntr=0.3,0.1

Type RM Length L Ch R = 1 ,66350   ,394,394,394
BEGIN DESCRIPTION:
Turtle Creek 105.0
END DESCRIPTION:
XS GIS Cut Line= 3
      1900968.62     13900850.21        1900125.       13899975.
      1899725.01     13899175.02
#Sta/Elev= 30
  3784.4 1756.05    4597 1725.43  4943.5 1721.42  4996.5 1704.27  5002.8 1704.27
  5003.1 1700.92  5004.1 1700.42  5041.7 1700.92  5058.7 1705.29  5126.1 1707.34
  5187.3 1705.08  5215.2 1712.23  5259.9 1711.39  5299.1 1716.06  5349.4 1728.86
  5366.2 1735.49  5371.7 1733.38  5388.5 1739.97  5394.1  1738.4  5410.9 1743.67
  5416.5 1742.48  5433.2 1747.64    5453 1749.83  5503.1 1759.02    5545 1763.61
  5595.4 1773.61  5656.8  1793.3  5715.5 1797.73  5796.6 1811.06  5894.4  1836.7
#Mann= 6 ,-1 , 0
  3784.4     .07       0  5003.1     .05       0  5041.7     .07       0
  5126.1      .1       0    5453     .07       0  5503.1      .1       0
Bank Sta=5003.1,5041.7
XS Rating Curve= 0 ,0
Exp/Cntr=0.3,0.1

Type RM Length L Ch R = 1 ,65956   ,701,701,701
BEGIN DESCRIPTION:
Turtle Creek 104.0
END DESCRIPTION:
XS GIS Cut Line= 3
      1901122.53     13900404.52      1900414.96     13899742.16
      1899724.98     13898874.97
#Sta/Elev= 30
  3990.7 1741.09  4512.1 1722.27  4781.2 1719.03  4788.1 1727.02  4802.2 1718.84
  4909.4 1718.58  4929.7 1718.69  4982.3 1709.26  4994.1 1705.68  4995.6 1700.63
  4996.6 1700.13  5034.3 1700.63  5174.2 1707.35  5213.5 1704.55    5236 1706.62
  5271.2 1726.01  5285.6 1737.58    5300 1755.18  5314.1 1763.59  5353.9 1765.33
  5463.4 1774.66  5527.5 1785.55  5548.3  1792.7  5584.2 1796.79  5626.8 1804.47
  5705.3 1806.66  5734.1 1812.21  5862.3 1847.39  6017.6 1900.42  6068.1 1911.64
#Mann= 8 ,-1 , 0
  3990.7     .07       0  4909.4      .1       0  4982.3     .07       0
  4995.6     .05       0  5034.3     .07       0  5174.2      .1       0
  5353.9     .07       0  5584.2      .1       0
Bank Sta=4995.6,5034.3
XS Rating Curve= 0 ,0
Exp/Cntr=0.3,0.1

Type RM Length L Ch R = 1 ,65255   ,1134,1134,1134
BEGIN DESCRIPTION:
Turtle Creek 103.0
END DESCRIPTION:
XS GIS Cut Line= 3
       1901257.4     13900301.17        1900775.       13899275.
        1899975.       13898775.
#Sta/Elev= 30
  3870.2 1740.86    3872  1740.7  3907.9 1740.79  3930.7 1737.43  4101.3  1728.1
    4386 1720.86  4506.9 1706.46  4562.1 1712.11  4716.8 1712.29  4875.9 1708.44
  4937.8 1703.27  4947.7 1698.01  4948.7 1697.51  4986.5 1698.01  5048.3 1702.04
  5054.2 1709.08  5069.5 1714.33  5075.4  1724.3  5100.2 1728.61  5142.7 1733.87
  5238.5 1738.97  5525.9 1751.85  5608.7 1759.46  5693.4 1766.69  5808.9 1786.13
  5824.3 1792.32  5845.5 1795.62  5903.3  1815.4  5918.6 1824.12  5947.5 1834.53
#Mann= 7 ,-1 , 0
  3870.2    .035       0    3872     .07       0  4947.7     .05       0
  4986.5     .07       0  5100.2      .1       0  5238.5     .07       0
  5608.7      .1       0
Bank Sta=4947.7,4986.5
XS Rating Curve= 0 ,0
Exp/Cntr=0.3,0.1

Type RM Length L Ch R = 1 ,64121   ,501,501,501
BEGIN DESCRIPTION:
Turtle Creek 102.0
END DESCRIPTION:
XS GIS Cut Line= 3
      1902124.99       13899375.        1901725.       13899275.
      1900425.04     13898875.01
#Sta/Elev= 30
  4588.1 1783.41  4611.3 1780.76  4688.6 1755.75  4693.7 1755.76  4729.8 1739.92
  4742.7 1737.02  4858.7 1727.84  4866.1 1725.72  4907.6 1719.51  4917.9 1705.36
  4928.2 1699.72  4959.9 1699.08  5002.4 1698.55  5003.4 1698.05  5041.5 1698.55
  5063.2 1701.72  5094.6 1700.62    5126  1703.7  5146.9 1703.79  5185.5 1708.59
  5218.2 1710.38    5294 1711.83    5398 1717.18  5528.1 1717.27    5566 1719.21
  5711.9 1717.29    5956 1724.27  5994.4 1724.24    6247 1736.78  6360.5 1742.82
#Mann= 7 ,-1 , 0
  4588.1     .07       0  4866.1      .1       0  4959.9     .07       0
  5002.4     .05       0  5041.5     .07       0    5956      .1       0
    6247     .07       0
Bank Sta=5002.4,5041.5
XS Rating Curve= 0 ,0
Exp/Cntr=0.3,0.1

Type RM Length L Ch R = 1 ,63620   ,444,444,444
BEGIN DESCRIPTION:
Turtle Creek 101.0
END DESCRIPTION:
XS GIS Cut Line= 3
      1902075.03       13898925.        1901675.       13898875.
      1900074.97       13898775.
#Sta/Elev= 30
  4604.9 1782.62  4625.1 1779.65  4642.7 1771.82  4685.6 1767.16  4735.9 1755.73
    4780    1740    4804  1730.7  4816.6 1730.48    4867 1714.82  4884.6 1700.59
  4893.5 1700.72  4998.5 1698.37  4999.5 1697.87  5037.7 1698.37  5038.1 1701.26
  5090.7 1701.18  5138.3 1709.22  5258.5 1717.37  5448.9 1716.06  5639.3 1721.56
  5753.1  1721.5  5784.6 1721.29  5821.2 1721.44  5919.8 1722.83    6010  1730.2
  6170.5 1734.72  6270.5 1739.58  6416.4 1752.89  6533.5 1774.02  6611.2 1795.25
#Mann= 10 ,-1 , 0
  4604.9     .07       0    4780    .033       0  4893.5     .07       0
  4998.5     .05       0  5037.7     .07       0  5753.1      .1       0
  5784.6     .07       0  5821.2      .1       0  6170.5     .07       0
  6416.4      .1       0
Bank Sta=4998.5,5037.7
XS Rating Curve= 0 ,0
Exp/Cntr=0.3,0.1

Type RM Length L Ch R = 1 ,63176   ,645,645,645
BEGIN DESCRIPTION:
Turtle Creek 100.0
END DESCRIPTION:
XS GIS Cut Line= 3
       1902119.7     13898466.07      1901697.84     13898490.81
      1901224.99       13898475.
#Sta/Elev= 30
  4554.5 1763.49  4617.9 1761.19    4623 1762.35  4659.4 1762.11  4749.5 1758.02
  4769.6 1755.57  4779.6 1752.24  4788.5 1746.86  4793.5 1747.93  4799.6 1740.73
  4859.7 1706.44  4869.7 1702.41  4889.8 1698.16  4899.8 1693.57  4907.2 1692.73
  4919.8 1695.25  4990.4 1695.62  5009.9 1694.08    5040 1694.66  5060.4 1691.61
  5061.4 1691.11  5099.6 1691.61    5100 1698.54    5110 1698.75    5130 1706.24
    5150 1710.97    5180 1713.34  5304.9 1714.47  5447.3  1716.6  5450.2 1716.61
#Mann= 7 ,-1 , 0
  4554.5     .07       0  4907.2    .033       0  4990.4     .07       0
  5060.4     .05       0  5099.6     .07       0  5304.9    .035       0
  5447.3     .07       0
Bank Sta=5060.4,5099.6
XS Rating Curve= 0 ,0
Exp/Cntr=0.3,0.1

Type RM Length L Ch R = 1 ,62531   ,545,545,545
BEGIN DESCRIPTION:
Turtle Creek 99.0
END DESCRIPTION:
XS GIS Cut Line= 3
      1902075.02     13898375.02        1901675.       13897925.
      1900958.77     13897842.22
#Sta/Elev= 30
  4393.5 1757.91  4414.8 1758.14  4443.3 1755.51  4457.5 1748.22  4513.9 1742.58
  4592.1 1725.63  4627.2 1719.84  4690.8 1702.66  4714.2  1700.8  4782.8 1695.04
  4804.5 1695.57  4854.4 1693.76  4903.2  1692.1  4939.2 1692.61  4953.4 1689.15
  4972.7 1687.83  4973.7 1687.33  5011.9 1687.83  5024.1 1688.13  5045.9  1688.9
  5066.1 1699.62  5076.1 1701.23  5086.2 1706.11  5096.3 1713.11  5136.5 1713.81
  5146.6 1715.09  5217.7  1715.7  5396.5 1713.91  5711.2 1714.21  5716.6 1714.39
#Mann= 8 ,-1 , 0
  4393.5     .07       0  4714.2    .035       0  4854.4     .07       0
  4972.7    .035       0  5011.9     .07       0  5024.1     .07       0
  5396.5    .035       0  5711.2     .07       0
Bank Sta=4972.7,5011.9
XS Rating Curve= 0 ,0
Exp/Cntr=0.3,0.1

Type RM Length L Ch R = 1 ,61986   ,562,562,562
BEGIN DESCRIPTION:
Turtle Creek 98.0
END DESCRIPTION:
XS GIS Cut Line= 3
      1902374.99     13898274.99        1901925.       13897475.
      1901116.54     13897249.07
#Sta/Elev= 30
  4082.1 1761.96  4155.1 1754.16  4212.5 1742.88    4323 1723.55  4376.3 1717.42
  4506.6 1711.59  4669.5 1708.73  4690.2 1709.12  4731.9 1706.08  4765.1 1705.15
  4770.8 1702.82  4802.7 1698.72  4808.4 1696.47  4851.8 1694.52  4932.7 1686.44
    4977 1685.68  4977.5 1683.25  4978.5 1682.75  5016.7 1683.25    5017 1685.74
  5031.1 1684.02  5041.5 1685.14  5062.3 1692.18  5090.5 1698.46  5124.6 1702.54
  5145.3  1708.3    5164 1710.68    5195 1711.89  5578.6 1711.95  5839.4 1714.71
#Mann= 8 ,-1 , 0
  4082.1      .1       0  4212.5     .07       0  4669.5    .035       0
  4731.9     .07       0  4977.5     .05       0  5016.7     .07       0
    5195    .035       0  5578.6     .07       0
Bank Sta=4977.5,5016.7
XS Rating Curve= 0 ,0
Exp/Cntr=0.3,0.1

Type RM Length L Ch R = 1 ,61424   ,536,536,536
BEGIN DESCRIPTION:
Turtle Creek 97.0
END DESCRIPTION:
XS GIS Cut Line= 3
      1902702.19     13897796.27        1902225.       13897025.
      1901674.39     13896774.66
#Sta/Elev= 30
    4093 1734.75  4156.7 1730.54  4172.1 1723.48  4200.3 1715.26  4245.3 1710.87
  4303.3 1708.09    4376 1707.68  4564.9 1708.76  4681.5  1705.7  4729.9 1700.91
  4803.2 1699.57  4891.8 1687.37  4897.7 1684.23  4905.9 1683.11  4928.5 1682.24
  4949.7 1683.48  4972.5 1681.87  4973.5 1681.37  5012.1 1681.87  5031.8 1688.13
  5060.4 1690.48  5088.9 1697.83  5129.6 1701.78  5135.1 1704.15  5181.2 1705.48
  5197.7 1710.08  5417.3 1710.96  5445.9 1709.27  5461.3 1711.29  5604.8 1711.67
#Mann= 4 ,-1 , 0
    4093     .07       0    4376    .035       0  4972.5    .035       0
  5012.1    .035       0
Bank Sta=4972.5,5012.1
XS Rating Curve= 0 ,0
Exp/Cntr=0.3,0.1

Type RM Length L Ch R = 1 ,60888   ,540,540,540
BEGIN DESCRIPTION:
Turtle Creek 96.0
END DESCRIPTION:
XS GIS Cut Line= 4
      1902741.95     13897777.59        1902675.       13897175.
        1902625.       13896725.      1903074.98     13895925.04
#Sta/Elev= 30
  3948.4 1731.59  3981.2 1729.97  4041.6 1722.12  4091.9 1711.57    4122 1708.56
  4372.9 1706.83  4408.3  1707.1  4507.7 1705.31  4584.9 1703.62  4846.5 1690.35
  4954.5 1676.56  4955.5 1676.06  5000.1 1676.56  5021.2 1678.08  5039.8 1687.77
    5053 1693.57  5058.8 1691.55  5064.8 1705.42  5074.7 1708.92  5114.8    1708
  5225.7 1707.12  5447.6 1706.54  5528.6 1711.01  5549.4 1715.48  5609.5 1733.29
  5615.6 1738.14  5647.1 1752.59  5793.1 1798.74  5799.1 1802.95  5925.3 1854.06
#Mann= 10 ,-1 , 0
  3948.4     .07       0  4372.9    .035       0  4408.3     .07       0
  4507.7    .035       0  4954.5     .05       0  5000.1    .035       0
  5039.8      .1       0  5114.8     .07       0  5225.7    .035       0
  5549.4      .1       0
Bank Sta=4954.5,5000.1
XS Rating Curve= 0 ,0
Exp/Cntr=0.3,0.1

Type RM Length L Ch R = 1 ,60348   ,518,518,518
BEGIN DESCRIPTION:
Turtle Creek 95.0
END DESCRIPTION:
XS GIS Cut Line= 4
      1902820.77     13897790.52        1902975.       13897225.
        1903125.       13896675.      1903874.99       13896225.
#Sta/Elev= 30
  3847.9 1728.42  4081.7 1709.14  4326.7 1705.11  4427.8 1705.24  4553.6 1696.53
  4776.1 1690.27  4848.7 1683.03  4907.4 1683.44  4989.1 1673.39  4990.1 1672.89
  5034.7 1673.39  5039.2  1704.4  5132.5 1704.57  5282.1 1705.53  5441.5 1711.87
  5489.2 1717.67  5552.3  1731.5  5637.8 1770.93  5696.1 1807.93  5711.7 1811.73
  5717.5 1817.72  5727.2  1819.7  5738.9 1830.78  5748.6 1833.54  5754.4 1843.17
    5770 1853.04  5806.9 1892.09  5820.5 1911.12  5855.5 1924.21  5878.8 1924.34
#Mann= 8 ,-1 , 0
  3847.9     .07       0  4326.7    .035       0  4427.8     .07       0
  4553.6    .035       0  4989.1     .05       0  5034.7    .035       0
  5132.5    .035       0  5489.2      .1       0
Bank Sta=4989.1,5034.7
XS Rating Curve= 0 ,0
Exp/Cntr=0.3,0.1

Type RM Length L Ch R = 1 ,59830   ,620,620,620
BEGIN DESCRIPTION:
Turtle Creek 94.0
END DESCRIPTION:
XS GIS Cut Line= 4
      1903204.81     13897853.64        1903425.       13897275.
      1903593.48     13896832.25      1903975.03     13896374.96
#Sta/Elev= 30
  3915.3 1708.96  4138.5 1703.67  4494.6 1702.33  4565.6 1697.72  4598.6 1694.32
  4714.1 1691.11  4744.2  1686.2  4834.5  1684.2  4866.1 1678.65  4908.8 1677.25
  4944.9 1671.96  4946.2 1671.62  4947.2 1671.12  4991.8 1671.62  4993.8 1698.68
  4999.1 1703.69  5070.7 1702.45  5177.7 1705.64  5255.5 1717.23  5298.4  1729.4
  5341.4 1746.09  5440.3 1804.35  5489.8 1839.45  5518.4 1862.52  5532.7 1879.08
  5539.2 1881.19    5547 1902.19  5553.5 1909.76  5575.7 1924.11  5603.7 1926.92
#Mann= 6 ,-1 , 0
  3915.3     .07       0  4565.6    .035       0  4944.9     .07       0
  4946.2     .05       0  4991.8     .07       0  5177.7      .1       0
Bank Sta=4946.2,4991.8
XS Rating Curve= 0 ,0
Exp/Cntr=0.3,0.1

Type RM Length L Ch R = 1 ,59210   ,561,561,561
BEGIN DESCRIPTION:
Turtle Creek 93.0
END DESCRIPTION:
XS GIS Cut Line= 4
      1903447.97     13898164.54        1903825.       13897525.
        1904025.       13897175.      1904275.01     13896624.97
#Sta/Elev= 30
  3859.1 1706.21  4119.4 1701.08  4569.4 1701.88  4652.6 1702.35  4705.2 1698.49
  4749.1 1692.63  4792.3 1691.42  4820.3 1686.78  4872.9 1682.48  4888.7 1683.65
  4937.7  1679.3  4962.8 1673.63  4973.8 1670.99  4974.8 1670.49  5019.5 1670.99
  5036.5  1672.9  5048.6 1677.24  5070.5 1698.22  5120.5 1701.96  5180.4 1712.49
  5191.4 1724.57  5227.1 1740.23  5268.2 1757.45  5323.2 1775.68  5404.5 1810.54
  5531.9  1876.1  5542.9  1880.2  5564.8 1891.89  5576.9 1902.09  5608.8 1904.87
#Mann= 7 ,-1 , 0
  3859.1     .07       0  4569.4    .035       0  4962.8     .07       0
  4973.8     .05       0  5019.5     .07       0  5120.5     .07       0
  5227.1      .1       0
Bank Sta=4973.8,5019.5
XS Rating Curve= 0 ,0
Exp/Cntr=0.3,0.1

Type RM Length L Ch R = 1 ,58649   ,495,495,495
BEGIN DESCRIPTION:
Turtle Creek 92.0
END DESCRIPTION:
XS GIS Cut Line= 4
      1903416.74     13898352.02        1904125.       13897675.
        1904475.       13897475.        1904575.     13897075.02
#Sta/Elev= 30
  3617.2 1732.12  3698.6 1714.12  3804.9 1704.72  4080.7 1700.32  4438.3 1700.51
  4685.5 1700.45  4744.6 1696.54  4771.9 1691.11  4884.2 1683.46  4927.4 1678.52
  4933.2 1674.72    4949 1673.89  4963.6 1670.11  4964.6 1669.61  5009.3 1670.11
  5064.5 1671.18  5092.9 1676.49  5099.9 1681.71  5113.5 1694.91    5147 1698.47
  5200.5 1716.31  5216.6 1724.53  5224.3 1730.82  5229.5 1731.82  5265.5  1751.2
  5270.7 1751.45  5288.7 1759.37  5311.9 1764.94  5371.2 1786.85  5412.4 1789.96
#Mann= 6 ,-1 , 0
  3617.2     .07       0  4438.3    .035       0  4963.6    .035       0
  5009.3    .035       0  5099.9    .094       0  5200.5      .1       0
Bank Sta=4963.6,5009.3
XS Rating Curve= 0 ,0
Exp/Cntr=0.3,0.1

Type RM Length L Ch R = 1 ,58154   ,568,568,568
BEGIN DESCRIPTION:
Turtle Creek 91.0
END DESCRIPTION:
XS GIS Cut Line= 5
      1904427.14     13898950.97      1904625.05     13898294.76
      1904855.01     13897764.99       1904906.2     13897663.88
        1904725.     13897074.99
#Sta/Elev= 30
  3655.6 1738.11  3732.3 1729.33  3808.7 1710.78  3841.6 1707.46  4316.7 1698.19
  4511.5 1694.78  4512.1 1694.77  4775.9 1696.11  4828.2 1688.07  4971.4 1673.57
  4976.4 1667.02  4977.4 1666.52  5022.1 1667.02  5087.6 1671.48  5112.2 1679.56
  5122.2 1683.52  5145.8 1683.01    5153 1689.28  5158.2 1685.91  5166.7 1692.06
  5177.2 1694.45  5216.1 1695.22  5344.6 1698.46  5392.3 1702.24    5424 1713.56
  5522.4 1752.82  5528.3  1757.6  5548.1 1763.24  5616.6 1785.83    5648 1789.66
#Mann= 11 ,-1 , 0
  3655.6     .07       0  4316.7    .035       0  4511.5     .07       0
  4512.1    .035       0  4976.4    .035       0  5022.1    .035       0
  5112.2    .035       0  5122.2    .094       0  5216.1    .035       0
    5424     .07       0  5548.1      .1       0
Bank Sta=4976.4,5022.1
XS Rating Curve= 0 ,0
Exp/Cntr=0.3,0.1

Type RM Length L Ch R = 1 ,57586   ,566,566,566
BEGIN DESCRIPTION:
Turtle Creek 90.0
END DESCRIPTION:
XS GIS Cut Line= 4
        1905329.     13898804.41        1905375.       13897925.
        1905375.       13897525.      1905182.21       13897019.
#Sta/Elev= 30
  4119.4 1716.28  4237.4 1711.69  4419.2 1705.95  4439.2 1706.17  4469.3 1704.35
  4535.3 1703.24  4633.7 1700.69    4732 1698.61  4799.7 1698.44  4837.5 1696.48
  4849.8 1697.09  4859.8 1688.55  4899.6 1677.43  4919.9 1674.27  4939.9 1668.31
    4970 1668.72  4980.3 1665.77  4987.1 1665.62  4988.1 1665.12    5033 1665.62
    5060 1669.55    5070 1669.98    5090 1676.71    5110 1686.63    5120  1688.3
  5223.8 1692.92  5524.7 1696.25  5809.6 1697.32  5889.2 1699.52  5941.5 1703.27
#Mann= 10 ,-1 , 0
  4119.4      .1       0  4237.4    .035       0  4535.3     .07       0
  4633.7    .035       0    4732     .07       0  4837.5      .1       0
  4980.3     .07       0  4987.1     .05       0    5033     .07       0
  5223.8    .035       0
Bank Sta=4987.1,5033
XS Rating Curve= 0 ,0
Exp/Cntr=0.3,0.1

Type RM Length L Ch R = 1 ,57020   ,539,539,539
BEGIN DESCRIPTION:
Turtle Creek 89.0
END DESCRIPTION:
XS GIS Cut Line= 3
      1905844.17     13898347.45        1905875.       13897925.
      1905580.57     13897019.97
#Sta/Elev= 30
  4581.7 1699.93  4764.6 1697.19  4874.9  1697.2    4895 1694.54    4905 1694.27
    4915 1692.32    4918 1688.72  4925.1 1680.21  4933.3 1672.51  4938.3 1674.67
  4945.1 1671.76  4965.2 1667.57  4972.3 1663.32  4973.3 1662.82  5018.3 1663.32
  5036.8 1663.97  5047.3 1666.74  5066.6 1668.34  5085.1 1671.62  5090.4 1671.83
  5110.4  1677.3    5142 1679.79    5163 1682.56  5173.5 1684.17  5186.2 1687.48
  5212.9 1690.33  5226.1 1689.61  5457.5 1694.22  5909.6 1695.77    5957 1696.07
#Mann= 7 ,-1 , 0
  4581.7      .1       0    4918     .07       0  4972.3     .05       0
  5018.3     .07       0  5066.6     .07       0  5226.1    .035       0
  5909.6     .07       0
Bank Sta=4972.3,5018.3
XS Rating Curve= 0 ,0
Exp/Cntr=0.3,0.1

Type RM Length L Ch R = 1 ,56481   ,705,705,705
BEGIN DESCRIPTION:
Turtle Creek 88.0
END DESCRIPTION:
XS GIS Cut Line= 3
      1906525.02     13898125.03        1906325.       13897775.
      1905884.29     13897251.05
#Sta/Elev= 30
    4592 1697.53  4615.1 1696.58  4664.7 1697.02  4680.6 1696.04  4841.7 1695.37
    4885 1695.08  4937.6 1693.62    4944 1683.34  4949.8 1678.83  4959.9 1669.06
  4965.6 1666.65  4987.2 1664.94  4992.3  1663.7    5043 1663.58    5044 1663.08
    5088 1663.08    5089 1663.58  5094.6 1666.24  5107.2 1668.28  5115.5 1669.36
  5123.2 1671.85  5158.4 1676.15    5164 1677.87  5179.2 1681.02  5201.3 1686.99
  5226.8 1689.24  5243.4 1690.82  5257.3 1690.52  5363.9 1692.18  5679.8 1693.55
#Mann= 8 ,-1 , 0
    4592     .07       0  4841.7    .035       0    4944     .07       0
    5043     .05       0    5089     .07       0  5107.2    .035       0
    5164     .07       0  5226.8    .035       0
Bank Sta=5043,5089
XS Rating Curve= 0 ,0
Exp/Cntr=0.3,0.1

Type RM Length L Ch R = 1 ,55776   ,390,390,390
BEGIN DESCRIPTION:
Turtle Creek 87.0
END DESCRIPTION:
XS GIS Cut Line= 3
      1906479.22     13898680.16      1906922.54     13897650.59
      1906995.74     13896870.78
#Sta/Elev= 30
  3853.3 1703.05    4142 1692.94    4240 1692.45  4281.6 1695.19  4415.6 1696.96
  4591.2 1694.89  4691.8 1690.26  4766.8 1688.72  4811.6 1685.36  4866.4 1674.38
  4947.8 1666.23  4955.6 1661.96  4956.6 1661.46  5004.2 1661.96  5071.1 1663.67
  5080.3 1664.01  5100.4 1672.59  5140.6  1682.8  5269.3 1695.91  5281.5  1698.8
  5375.9 1721.16  5401.7 1729.83  5451.9 1742.14  5484.6 1753.37  5572.5 1790.69
  5588.3    1801    5697 1858.88    5703 1865.19  5752.9 1888.09  5757.5 1888.09
#Mann= 7 ,-1 , 0
  3853.3     .07       0  4691.8    .035       0  4955.6    .035       0
  5004.2    .035       0  5071.1      .1       0  5269.3     .07       0
  5281.5      .1       0
Bank Sta=4955.6,5004.2
XS Rating Curve= 0 ,0
Exp/Cntr=0.3,0.1

Type RM Length L Ch R = 1 ,55386   ,520,520,520
BEGIN DESCRIPTION:
Turtle Creek 86.0
END DESCRIPTION:
XS GIS Cut Line= 4
      1906723.98     13898701.04      1907085.12     13898262.55
        1907275.       13897575.        1907125.       13896825.
#Sta/Elev= 30
  3726.6 1698.69  3923.5 1691.32  4591.6 1688.61  4690.1 1688.02  4724.4 1685.53
  4779.7 1680.11  4821.2 1670.79  4915.9 1663.35  4966.5 1661.41  4967.5 1660.91
  5015.1 1661.41  5048.7 1670.12  5069.1 1684.22  5079.3 1687.28    5118 1690.94
  5191.5 1704.39  5242.5    1720  5283.3  1736.2  5334.3  1750.8  5344.5 1749.32
  5385.3 1757.35  5395.5  1755.7  5446.5 1766.46  5477.1  1776.2  5538.2  1803.6
  5568.8  1819.9    5630 1853.02  5721.8 1906.85  5742.2 1915.25  5772.8 1921.62
#Mann= 6 ,-1 , 0
  3726.6     .07       0  4591.6    .035       0  4915.9     .07       0
  4966.5     .05       0  5015.1     .07       0    5118      .1       0
Bank Sta=4966.5,5015.1
XS Rating Curve= 0 ,0
Exp/Cntr=0.3,0.1

Type RM Length L Ch R = 1 ,54866   ,426,426,426
BEGIN DESCRIPTION:
Turtle Creek 85.0
END DESCRIPTION:
XS GIS Cut Line= 4
      1906812.54     13898742.68      1907316.46     13898309.66
        1907725.       13897575.      1907924.98     13897225.03
#Sta/Elev= 30
  3494.8  1695.7  3671.9 1692.27  3941.8  1691.1  4289.3 1686.99  4633.7 1685.59
  4713.8 1680.27  4736.7 1676.45  4758.5 1670.59  4764.2 1671.13  4781.7 1667.43
  4829.4 1665.66  4858.8 1661.91  4859.8 1661.41  4907.5 1661.91  4991.8 1662.35
  5051.2 1668.29  5057.4 1671.89  5066.8 1674.49  5072.5 1671.26  5088.4 1675.72
  5094.1  1681.8  5131.6  1693.3  5196.3  1726.3  5249.6 1746.84    5287 1752.88
  5299.3 1757.29  5314.4  1759.9  5345.3 1763.11  5373.4 1771.88  5402.9  1774.4
#Mann= 6 ,-1 , 0
  3494.8     .07       0  4289.3    .035       0  4781.7     .07       0
  4858.8     .05       0  4907.5     .07       0  5051.2      .1       0
Bank Sta=4858.8,4907.5
XS Rating Curve= 0 ,0
Exp/Cntr=0.3,0.1

Type RM Length L Ch R = 1 ,54440   ,262,262,262
BEGIN DESCRIPTION:
Turtle Creek 84.0
END DESCRIPTION:
XS GIS Cut Line= 4
      1907622.34     13898886.84      1908107.32     13897742.68
      1908152.77     13897498.59        1908025.     13897275.01
#Sta/Elev= 30
  3680.1 1690.35  3730.9 1689.36  3812.8 1688.44    3845 1684.32  3964.5 1684.48
  3997.1 1686.94  4190.8 1684.05    4540 1685.64  4768.4 1681.47  4844.3 1674.83
  4887.7 1661.89    4965 1661.71    4966 1661.21  5013.7 1661.71  5050.3 1663.19
  5113.7 1666.68  5152.6 1676.91  5157.7 1675.43  5185.8 1687.06  5194.7 1692.27
  5200.4 1691.73  5216.3 1701.02    5222 1700.09  5253.7 1715.03  5259.4 1715.17
    5281 1726.19  5296.9 1742.01  5318.5 1750.28  5324.9 1756.97  5428.6 1769.94
#Mann= 9 ,-1 , 0
  3680.1     .07       0  3730.9    .035       0  3812.8     .07       0
  4190.8    .035       0  4768.4     .07       0    4965    .033       0
  5013.7     .07       0  5050.3     .07       0  5185.8      .1       0
Bank Sta=4965,5013.7
XS Rating Curve= 0 ,0
Exp/Cntr=0.3,0.1

Type RM Length L Ch R = 1 ,54178   ,353,353,353
BEGIN DESCRIPTION:
Turtle Creek 83.1
END DESCRIPTION:
XS GIS Cut Line= 4
       1908299.4     13898287.71      1908328.04      13897795.5
      1908338.46     13897589.77      1908283.77     13897144.45
#Sta/Elev= 30
  4434.9  1684.3  4447.1 1683.97  4577.9 1683.93  4776.1 1681.19  4801.4 1679.42
  4878.4 1674.07    4932 1664.99  4965.1 1661.64  5004.2  1661.5  5005.2    1661
  5052.9  1661.5  5112.8 1666.71  5158.9 1673.82  5198.8 1682.19  5203.8 1681.76
  5219.3  1687.1  5239.5 1691.83  5258.9 1699.52  5269.7 1705.08  5285.1 1716.15
  5290.2 1715.54  5299.9 1719.25  5320.1 1723.44  5360.4 1726.45  5371.5 1728.79
  5447.8 1732.71  5452.8 1734.64  5501.4 1734.31  5529.1 1739.91  5582.6 1746.59
#Mann= 9 ,-1 , 0
  4434.9     .07       0  4447.1    .035       0  4776.1     .07       0
  4801.4    .035       0    4932     .07       0  5004.2     .05       0
  5052.9     .07       0  5112.8     .07       0  5258.9      .1       0
Bank Sta=5004.2,5052.9
XS Rating Curve= 0 ,0
Exp/Cntr=0.3,0.1

Type RM Length L Ch R = 1 ,53825   ,420,420,420
BEGIN DESCRIPTION:
Turtle Creek 83.0
END DESCRIPTION:
XS GIS Cut Line= 4
      1908578.32     13899097.07      1908641.16     13897784.21
      1908630.61     13897653.97      1908424.98     13897324.97
#Sta/Elev= 30
  3625.7 1693.55  4038.2 1683.55  4081.2 1681.52  4188.4 1671.33  4358.6 1680.63
  4408.7 1681.79  4628.9 1680.53  4869.2 1669.73  4942.2 1663.37  4954.4 1658.46
  4969.4 1656.09  5015.2 1655.72  5016.2 1655.22  5063.9 1655.72  5073.6 1656.31
    5089  1659.6    5168 1661.56    5247 1667.81  5256.4  1669.6  5277.7 1684.93
  5283.5 1692.24    5293 1697.84  5298.9 1699.32  5305.4 1703.53  5314.2 1706.44
  5335.4 1708.98  5393.2 1708.34  5414.4  1713.4  5429.8 1718.74  5458.7 1722.02
#Mann= 3 ,-1 , 0
  3625.7     .07       0  5015.2     .05       0  5063.9     .07       0
Bank Sta=5015.2,5063.9
XS Rating Curve= 0 ,0
Exp/Cntr=0.3,0.1

Type RM Length L Ch R = 1 ,53405   ,693,693,693
BEGIN DESCRIPTION:
Turtle Creek 82.0
END DESCRIPTION:
XS GIS Cut Line= 4
      1908659.52     13898980.41      1908953.92     13897772.98
      1908987.73     13897549.37      1908324.96     13896974.97
#Sta/Elev= 30
  3696.1 1690.94  4051.6  1684.3  4103.1 1680.13    4134  1667.7  4411.3 1679.42
  4574.2 1674.65  4691.4 1671.27  4719.1 1670.79  4885.4 1666.48  4958.6 1655.72
  4963.1 1655.62  4964.1 1655.12  5011.8 1655.62  5088.6 1655.79  5183.9 1664.31
  5361.6 1667.37  5404.3 1671.66  5432.8 1684.17  5439.4 1690.42  5453.7 1687.31
  5474.6 1697.24  5496.4 1694.41  5512.7 1695.98  5517.3 1698.15  5524.9  1693.1
  5560.1 1703.83  5666.4 1713.67  5709.2 1722.52  5749.1 1725.74  6042.1 1758.18
#Mann= 9 ,-1 , 0
  3696.1     .07       0  4574.2    .035       0  4691.4     .07       0
  4719.1    .035       0  4958.6     .07       0  4963.1     .05       0
  5011.8     .07       0  5512.7      .1       0  5749.1     .07       0
Bank Sta=4963.1,5011.8
XS Rating Curve= 0 ,0
Exp/Cntr=0.3,0.1

Type RM Length L Ch R = 1 ,52712   ,143,143,143
BEGIN DESCRIPTION:
Turtle Creek 81.0
END DESCRIPTION:
XS GIS Cut Line= 3
      1909398.14       13898866.        1909525.       13897825.
        1909225.       13897025.
#Sta/Elev= 30
  3951.3 1687.57  4018.8 1686.41  4227.3 1683.35  4399.1 1680.93  4466.9 1681.36
  4566.8 1679.43    4587 1676.23  4620.6 1668.07  4661.5 1661.94  4677.6 1658.61
  4706.8 1655.79    4794 1656.12  4965.6 1655.52  4966.6 1655.02  5014.3 1655.52
  5053.4  1658.6  5064.1 1662.81  5070.3 1672.34  5075.7 1666.24  5085.4 1674.33
  5095.2 1678.04  5100.6 1673.62  5106.8 1677.42  5117.5 1679.08  5149.5 1681.95
  5169.1 1680.91  5210.9 1679.13  5374.8 1677.97  5687.8 1682.08  5854.4 1690.28
#Mann= 12 ,-1 , 0
  3951.3    .035       0  4018.8     .07       0  4227.3    .035       0
  4399.1     .07       0  4620.6    .035       0  4661.5     .07       0
    4794    .033       0  4965.6    .033       0  5014.3    .033       0
  5169.1      .1       0  5374.8     .07       0  5687.8      .1       0
Bank Sta=4965.6,5014.3
XS Rating Curve= 0 ,0
Exp/Cntr=0.3,0.1

Type RM Length L Ch R = 1 ,52569   ,178,178,178
BEGIN DESCRIPTION:
Turtle Creek 80.2
END DESCRIPTION:
XS GIS Cut Line= 5
      1909458.25     13898805.91      1909591.06     13898053.31
        1909677.     13897756.44      1909601.48       13897233.
      1909270.89      13896685.4
#Sta/Elev= 30
  4099.1 1686.35  4166.1 1685.39  4344.1 1684.47  4487.1 1681.65    4625 1679.61
  4638.2 1678.57  4678.8 1671.35  4699.1 1666.17  4719.4    1664  4760.1 1661.03
  4802.7 1661.01    4821 1658.77  4881.5 1657.99  4896.7 1657.69    4924 1660.33
  4983.6 1655.28  4984.6 1654.78  5032.3 1655.28  5036.3  1657.1  5069.8 1660.69
  5080.3 1664.79  5087.8 1670.86    5101 1677.05    5189  1677.8  5277.2  1677.7
  5676.9  1676.1  5792.4 1677.08  6047.9  1683.9  6222.6 1692.52  6340.9  1700.1
#Mann= 10 ,-1 , 0
  4099.1     .07       0  4166.1    .035       0  4487.1     .07       0
  4881.5    .035       0  4983.6    .033       0  5032.3    .035       0
  5087.8      .1       0    5189     .07       0  5277.2      .1       0
  5676.9     .07       0
Bank Sta=4983.6,5032.3
XS Rating Curve= 0 ,0
Exp/Cntr=0.3,0.1

Type RM Length L Ch R = 1 ,52391   ,234,234,234
BEGIN DESCRIPTION:
Turtle Creek 80.1
END DESCRIPTION:
XS GIS Cut Line= 6
      1909516.17     13898790.06      1909774.79     13898026.79
      1909817.18     13897868.37      1909793.56     13897384.54
      1909765.67     13897143.72      1909333.99     13896639.22
#Sta/Elev= 30
    4153  1686.3  4354.5 1683.98  4432.9 1683.75  4567.4 1680.22  4622.9 1676.43
    4667 1668.53  4693.1  1665.5  4739.1 1663.88  4792.6 1659.61  4802.4 1657.95
  4819.6 1659.26  4844.6 1658.27  4865.8 1655.54  4881.6 1651.81  4907.8 1650.12
  4998.1 1649.17  4999.1 1648.67  5047.6 1649.17  5074.6 1654.18  5092.6 1666.54
  5105.7 1673.52    5122 1674.87  5206.4 1676.79  5294.9 1676.87  5501.9 1676.37
  5846.6 1674.45  5977.3 1675.56  6055.2 1679.03    6289 1685.26  6513.7 1696.91
#Mann= 7 ,-1 , 0
    4153     .07       0  4354.5    .035       0  4819.6     .07       0
  4998.1     .05       0  5047.6     .07       0  5294.9      .1       0
  5501.9     .07       0
Bank Sta=4998.1,5047.6
XS Rating Curve= 0 ,0
Exp/Cntr=0.3,0.1

Type RM Length L Ch R = 1 ,52157   ,565,565,565
BEGIN DESCRIPTION:
Turtle Creek 80.0
END DESCRIPTION:
XS GIS Cut Line= 5
        1910175.     13898374.99        1909975.       13898025.
        1909975.       13897625.      1909838.59     13897112.47
      1909438.75     13896665.89
#Sta/Elev= 30
  4603.7 1687.93  4670.6 1686.12  4741.9 1681.99  4751.3 1676.42    4757 1674.93
  4772.9 1661.59  4778.6 1661.12  4794.5 1654.74  4845.6 1654.94  4909.1 1648.92
  4910.1 1648.42  4959.1 1648.92  5046.8 1649.77  5056.8 1651.99  5076.8 1664.46
  5096.8 1668.09  5116.8 1669.93  5186.8 1674.12  5277.7 1676.26  5330.2 1676.42
  5376.8 1676.83  5544.7 1674.79  6043.9 1674.48  6129.2 1677.03  6135.9 1678.28
  6143.4 1677.59  6157.6 1678.93  6200.2 1679.06  6412.5  1684.5  6536.6 1690.22
#Mann= 5 ,-1 , 0
  4603.7     .07       0  4909.1     .05       0  4959.1     .07       0
  5277.7      .1       0  5330.2     .07       0
Bank Sta=4909.1,4959.1
XS Rating Curve= 0 ,0
Exp/Cntr=0.3,0.1

Type RM Length L Ch R = 1 ,51592   ,461,461,461
BEGIN DESCRIPTION:
Turtle Creek 79.0
END DESCRIPTION:
XS GIS Cut Line= 4
       1910585.6     13898896.11        1910475.       13898025.
      1909849.44     13897002.72      1909473.97     13896643.68
#Sta/Elev= 30
    4121 1702.54  4189.5 1700.12  4241.7 1698.26  4575.7 1691.55    4858 1682.15
  4868.1 1671.75  4876.6 1659.65  4881.6 1657.91  4888.2 1650.52  4948.7 1647.31
  4978.9 1648.81  4981.8 1647.25  4982.8 1646.75  5031.8 1647.25  5034.3    1649
  5101.6 1659.12  5196.4 1663.53  5312.5  1675.2  5339.7 1673.75  5370.5 1676.17
  5376.4 1674.71  5779.9 1674.99  5880.8 1674.94  5905.8 1675.16  6177.4 1673.94
  6411.3  1678.8  6418.4 1681.36  6425.3 1679.18  6595.1 1683.44  6717.1 1688.52
#Mann= 8 ,-1 , 0
    4121     .07       0  4189.5    .035       0  4241.7     .07       0
  4981.8     .05       0  5031.8     .07       0  5779.9    .035       0
  5880.8     .07       0  5905.8    .035       0
Bank Sta=4981.8,5031.8
XS Rating Curve= 0 ,0
Exp/Cntr=0.3,0.1

Type RM Length L Ch R = 1 ,51131   ,620,620,620
BEGIN DESCRIPTION:
Turtle Creek 78.0
END DESCRIPTION:
XS GIS Cut Line= 5
      1911053.58     13898924.46      1910844.11     13897927.97
      1910779.48     13897770.41      1909962.26     13896977.27
      1909505.24     13896565.58
#Sta/Elev= 30
  3925.9  1696.6  3972.7 1695.36  3984.2  1694.7  4201.3 1684.41  4450.1 1677.52
  4624.6 1676.74  4650.9  1674.4  4719.2 1673.57  4732.6  1671.6    4769 1673.84
  4774.1 1671.57  4813.8 1672.45  4818.9  1669.7  4853.8 1671.15  4863.6 1670.17
  4868.7 1666.32  4885.9 1662.13  4896.1 1658.04  4906.3 1651.56  4918.6 1649.46
  4965.6 1647.08  4966.6 1646.58  5015.6 1647.08  5060.6 1650.35  5084.6 1655.84
  5128.5 1659.28  5361.9 1673.32  6281.2 1674.03  6684.8 1681.68  6868.4  1688.4
#Mann= 7 ,-1 , 0
  3925.9     .07       0  3972.7    .035       0  3984.2     .07       0
  4450.1    .035       0  4853.8     .07       0  4965.6     .05       0
  5015.6     .07       0
Bank Sta=4965.6,5015.6
XS Rating Curve= 0 ,0
Exp/Cntr=0.3,0.1

Type RM Length L Ch R = 1 ,50511   ,415,415,415
BEGIN DESCRIPTION:
Turtle Creek 77.0
END DESCRIPTION:
XS GIS Cut Line= 3
      1911140.26     13898924.91        1911275.       13897575.
        1910724.      13894831.2
#Sta/Elev= 30
    3639 1697.05  3695.3 1694.06  3705.1 1693.45  3793.9 1689.67  3892.4 1685.05
    3991 1681.57  4211.7 1673.03  4768.3  1671.3  4814.7  1669.2  4842.2 1656.52
  4847.3 1660.62    4875 1649.41    4900 1647.09    4901 1646.59  4950.6 1647.09
  4972.8 1647.69  5036.4  1649.8  5179.2 1663.65  5250.6 1663.52  5342.4 1675.16
    5845    1675  6515.4 1674.44  7331.3 1685.05  7433.3 1690.12  7453.7 1696.23
  7474.1 1692.63  7525.1 1693.56  7611.6 1704.38  7759.2 1742.07  7794.2 1744.53
#Mann= 11 ,-1 , 0
    3639     .07       0  3695.3    .035       0  3705.1     .07       0
  3793.9    .035       0  3892.4     .07       0    3991    .035       0
  4768.3     .07       0    4900     .05       0  4950.6     .07       0
  4972.8     .07       0    5845    .045       0
Bank Sta=4900,4950.6
XS Rating Curve= 0 ,0
Exp/Cntr=0.3,0.1

Type RM Length L Ch R = 1 ,50096   ,537,537,537
BEGIN DESCRIPTION:
Turtle Creek 76.0
END DESCRIPTION:
XS GIS Cut Line= 5
        1911275.     13898925.01      1911618.73     13897593.05
      1911526.58     13897290.19      1911192.75     13896294.76
       1910786.5     13894862.44
#Sta/Elev= 30
  3494.7    1696  3547.9 1693.15  3648.7 1687.95  3763.2 1682.11  3800.1 1682.82
  3959.8 1675.12  4152.8 1671.01  4816.1 1668.62  4902.6 1663.43  4920.5 1654.04
  4941.3 1647.71  4948.2 1646.85  4949.2 1646.35  4998.8 1646.85  5065.1 1648.17
    5169 1658.78  5263.4 1668.33  5277.6 1669.04  5524.4 1671.06  6794.6 1674.72
  6995.3  1676.5    7311 1684.16  7411.1 1689.95  7431.9 1696.39  7463.1  1692.3
  7515.1  1695.6  7603.1  1709.3    7637 1719.69  7676.1 1725.85  7725.6 1741.63
#Mann= 13 ,-1 , 0
  3494.7     .07       0  3547.9    .035       0  3648.7     .07       0
  3800.1    .035       0  4816.1     .07       0  4941.3    .033       0
  4948.2    .033       0  4998.8    .033       0  5065.1     .07       0
    5169    .045       0  5263.4      .1       0  5277.6     .07       0
  5524.4    .045       0
Bank Sta=4948.2,4998.8
XS Rating Curve= 0 ,0
Exp/Cntr=0.3,0.1

Type RM Length L Ch R = 1 ,49559   ,647,647,647
BEGIN DESCRIPTION:
Turtle Creek 75.0
END DESCRIPTION:
XS GIS Cut Line= 5
      1911685.65     13899074.92       1912020.3     13897456.84
      1911984.67     13897138.64      1911292.22     13896238.33
      1910901.08     13894872.86
#Sta/Elev= 30
  3164.9 1706.01  3233.5 1699.19  3288.8 1699.13  3456.2 1687.45  3630.1 1679.68
  3949.6 1670.82  4523.8 1669.24  4553.6 1666.32  4601.3 1668.69  4808.9 1663.38
  4879.4 1648.81  4951.7 1646.28  4984.9 1645.26  4985.9 1644.76  5035.6 1645.26
  5040.4 1652.39  5060.6 1654.05  5087.6 1665.74    5155 1669.26  5536.7 1668.53
  6744.8 1673.05    7227 1681.05  7372.4  1688.4  7411.4 1691.57  7431.3 1696.31
  7439.9 1693.93  7472.9 1694.24  7608.2 1713.65  7639.4 1722.94  7693.6 1733.64
#Mann= 9 ,-1 , 0
  3164.9    .035       0  3456.2     .07       0  3949.6    .035       0
  4601.3     .07       0  4951.7    .033       0  4984.9    .033       0
  5035.6    .033       0    5155    .035       0  5536.7    .045       0
Bank Sta=4984.9,5035.6
XS Rating Curve= 0 ,0
Exp/Cntr=0.3,0.1

Type RM Length L Ch R = 1 ,48912   ,565,565,565
BEGIN DESCRIPTION:
Turtle Creek 74.0
END DESCRIPTION:
XS GIS Cut Line= 4
      1912630.86     13899010.23        1912575.       13897225.
      1912432.37     13896315.28      1911593.79     13894872.87
#Sta/Elev= 30
    3209 1707.02    3458 1694.79  3564.4 1688.65  3674.5 1684.59  3957.2 1677.77
  4061.2  1675.4  4320.2  1672.4  4594.9 1661.34    4695 1664.82  4832.6  1653.4
    4885 1651.07  4915.1 1645.48  4977.1 1645.02  4979.9 1644.95  4980.9 1644.45
  5030.6 1644.95  5045.7 1653.62  5077.7 1666.46  5177.8 1666.52  5678.1 1664.36
  5778.2 1664.34  5878.3  1664.1  5964.4 1665.28  6097.6 1664.15  6696.8 1669.37
  6814.4  1674.1  7070.9 1678.82  7223.4 1685.14  7237.3 1684.48  7584.4  1707.1
#Mann= 13 ,-1 , 0
    3209     .07       0    3458    .035       0  3957.2     .07       0
  4061.2    .035       0  4320.2     .07       0  4977.1    .033       0
  4979.9    .033       0  5030.6    .033       0  5077.7    .035       0
  5177.8    .045       0  5678.1    .035       0  5778.2    .045       0
  5878.3    .035       0
Bank Sta=4979.9,5030.6
XS Rating Curve= 0 ,0
Exp/Cntr=0.3,0.1

Type RM Length L Ch R = 1 ,48347   ,485,485,485
BEGIN DESCRIPTION:
Turtle Creek 73.1
END DESCRIPTION:
XS GIS Cut Line= 5
      1913200.44     13898337.18      1913075.44      13897298.1
      1913059.81     13897061.12      1913038.98     13896954.35
       1913156.3     13895174.96
#Sta/Elev= 30
  3826.2 1687.43  3843.4 1687.49  4590.5 1667.97  4684.5 1664.24  4734.9  1651.3
  4825.5 1651.22  4980.8 1641.87  4981.8 1641.37  5031.5 1641.87  5116.5  1642.8
  5193.1 1651.24  5248.5 1657.23  5268.5 1664.51  5434.9 1663.56  5491.7 1663.42
  5571.7 1663.04  5633.5 1662.87  5708.4 1662.06  5775.2 1661.36    5960 1658.19
    5970 1660.36    6411 1662.95  6541.3 1666.85  6755.7 1680.56  6761.7 1685.47
  6811.8 1691.69  6841.9 1698.47    6882 1712.18  6906.8 1716.99  7002.3 1745.09
#Mann= 12 ,-1 , 0
  3826.2    .035       0  3843.4     .07       0  4590.5    .035       0
  4980.8     .05       0  5031.5    .035       0  5193.1    .035       0
  5434.9     .07       0  5491.7    .035       0  5571.7     .07       0
  5633.5    .035       0  5708.4    .045       0  5775.2    .035       0
Bank Sta=4980.8,5031.5
XS Rating Curve= 0 ,0
Exp/Cntr=0.3,0.1

Type RM Length L Ch R = 1 ,47862   ,446,446,446
BEGIN DESCRIPTION:
Turtle Creek 73.0
END DESCRIPTION:
XS GIS Cut Line= 5
      1913701.55     13897631.38       1913598.7     13897393.15
        1913375.       13896875.      1913229.21      13896445.8
      1913255.25     13895284.34
#Sta/Elev= 30
  4180.3 1667.99  4372.4  1665.9  4680.2 1669.06    4745 1669.23  4895.7 1666.19
  4913.7 1648.51  4919.2 1645.19  4937.2 1643.14  4949.7 1636.26  4975.9 1635.49
  4976.9 1634.99  5026.9 1635.49  5099.2 1641.91  5110.4 1644.92  5120.3 1650.25
    5152 1652.25  5183.7 1651.71  5220.9 1658.04  5239.6 1661.23  5396.5 1662.44
  5638.3 1660.08  5658.3 1657.53  5688.3    1659  5728.3 1657.24  5768.3 1658.96
  6068.4  1660.5  6248.4 1665.75  6389.1 1673.88  6498.5 1687.71  6619.2 1710.69
#Mann= 7 ,-1 , 0
  4180.3     .07       0  4680.2    .035       0    4745     .07       0
  4975.9     .05       0  5026.9     .07       0  5110.4    .035       0
  5220.9     .07       0
Bank Sta=4975.9,5026.9
XS Rating Curve= 0 ,0
Exp/Cntr=0.3,0.1
