--- Verde Creek.prj (project) ---

Proj Title=Verde Creek Base Level Engineering
Current Plan=p01
Default Exp/Contr=0.3,0.1
English Units
Geom File=g01
Flow File=f01
Plan File=p01
Y Axis Title=Elevation
X Axis Title(PF)=Main Channel Distance
X Axis Title(XS)=Station
BEGIN DESCRIPTION:
Verde Creek
END DESCRIPTION:
DSS Export Rating Curves= 0
DSS Export Rating Curve Sorted= 0
DSS Export Volume Flow Curves= 0
DXF OffsetX= 0
DXF OffsetY= 0
DXF ScaleX= 1
DXF ScaleY= 10

--- Verde Creek.p01 (plan) ---

Plan Title=Multiple Run
Short Identifier=Multiple
Geom File=g01
Flow File=f01
Subcritical Flow
K Sum by GR= 0
Std Step Tol= 0.01
Critical Tol= 0.01
Num of Std Step Trials= 20
Max Error Tol= 0.3
Flow Tol Ratio= 0.001
Split Flow NTrial= 30
Split Flow Tol= 0.02
Split Flow Ratio= 0.02
Log Output Level= 0
Friction Slope Method= 1
Unsteady Friction Slope Method= 2
Unsteady Bridges Friction Slope Method= 1
Parabolic Critical Depth
Global Vel Dist=  1 , 1 , 1
Global Log Level= 0
CheckData=True
Encroach Param= -1, 0, 0, 0
BEGIN DESCRIPTION:
Multiple Run
END DESCRIPTION:

--- Verde Creek.f01 (steady flow) ---

Flow Title=Multiple
Number of Profiles=7
Profile Names=10-year,25-year,50-year,1pct_min,100-year,1pct_plu,500-year
River Rch & RM= Verde Creek,Reach-1,81743
    3130    5582    8022    5559   11092   22131   20941
River Rch & RM= Verde Creek,Reach-1,77700
    3621    6475    9321    6463   12896   25732   24384
River Rch & RM= Verde Creek,Reach-1,71467
    4261    7677   11106    7735   15434   30795   29447
River Rch & RM= Verde Creek,Reach-1,70575
    4494    8122   11772    8210   16381   32684   31350
River Rch & RM= Verde Creek,Reach-1,64701
    5863   10691   15587   10925   21798   43493   42141
River Rch & RM= Verde Creek,Reach-1,57617
    9914   18304   26911   18989   37888   75596   74215
River Rch & RM= Verde Creek,Reach-1,54989
   10793   19982   29435   20805   41512   82828   81590
River Rch & RM= Verde Creek,Reach-1,54448
   11460   21218   31256   22088   44072   87936   86580
River Rch & RM= Verde Creek,Reach-1,48311
   11594   21465   31618   22341   44577   88942   87551
River Rch & RM= Verde Creek,Reach-1,47219
   12922   23989   35402   25057   49996   99755   98512
River Rch & RM= Verde Creek,Reach-1,44484
   13053   24226   35748   25297   50474  100708   99412
River Rch & RM= Verde Creek,Reach-1,42315
   13185   24456   36070   25512   50904  101567  100158
River Rch & RM= Verde Creek,Reach-1,39564
   12844   23872   35251   24960   49802   99369   98251
River Rch & RM= Verde Creek,Reach-1,38497
   13779   25633   37874   26830   53533  106813  105697
River Rch & RM= Verde Creek,Reach-1,33427
   14143   26311   38877   27539   54948  109636  108476
River Rch & RM= Verde Creek,Reach-1,31246
   14177   26373   38968   27602   55074  109887  108711
River Rch & RM= Verde Creek,Reach-1,30249
   14179   26373   38964   27597   55062  109864  108667
River Rch & RM= Verde Creek,Reach-1,29597
   14204   26414   39019   27631   55132  110003  108770
River Rch & RM= Verde Creek,Reach-1,28475
   14170   26335   38886   27524   54918  109575  108247
River Rch & RM= Verde Creek,Reach-1,26274
   15434   28745   42511   30132   60121  119957  118823
River Rch & RM= Verde Creek,Reach-1,25095
   15574   29012   42909   30417   60690  121093  119968
River Rch & RM= Verde Creek,Reach-1,23540
   15571   28970   42810   30319   60494  120702  119358
River Rch & RM= Verde Creek,Reach-1,19194
   15702   29205   43149   30552   60959  121629  120216
River Rch & RM= Verde Creek,Reach-1,16467
   15695   29169   43074   30481   60818  121349  119803
River Rch & RM= Verde Creek,Reach-1,12584
   15839   29432   43456   30746   61346  122402  120799
River Rch & RM= Verde Creek,Reach-1,9763
   15926   29576   43652   30872   61597  122903  121187
River Rch & RM= Verde Creek,Reach-1,3226
   15950   29615   43703   30903   61660  123028  121272
River Rch & RM= Verde Creek,Reach-1,1410
   17519   32597   48176   34112   68063  135803  134211
Boundary for River Rch & Prof#=Verde Creek,Reach-1,1
Up Type=0
Dn Type=3
Dn Slope=0.005
Boundary for River Rch & Prof#=Verde Creek,Reach-1,2
Up Type=0
Dn Type=3
Dn Slope=0.005
Boundary for River Rch & Prof#=Verde Creek,Reach-1,3
Up Type=0
Dn Type=3
Dn Slope=0.005
Boundary for River Rch & Prof#=Verde Creek,Reach-1,4
Up Type=0
Dn Type=3
Dn Slope=0.005
Boundary for River Rch & Prof#=Verde Creek,Reach-1,5
Up Type=0
Dn Type=3
Dn Slope=0.005
Boundary for River Rch & Prof#=Verde Creek,Reach-1,6
Up Type=0
Dn Type=3
Dn Slope=0.005
Boundary for River Rch & Prof#=Verde Creek,Reach-1,7
Up Type=0
Dn Type=3
Dn Slope=0.005

--- Verde Creek.g01 (geometry) ---

Geom Title=Existing Conditions
Program Version=4.10

River Reach=Verde Creek     ,Reach-1
Reach XY= 30
        1912475.       13865125.      1913369.15     13865622.96
      1915168.68     13863883.06      1915702.12     13864151.49
      1917733.28     13870521.94      1919330.93     13869527.24
      1920773.53     13869721.46        1921275.       13869025.
      1921981.03     13871073.38      1924609.58     13869925.03
      1926741.14     13871424.45        1928625.     13870632.56
       1937373.5     13872678.62      1942830.04     13877469.92
      1944727.45     13877630.47      1946876.55     13879771.25
      1949805.01     13880275.06      1950981.19     13879432.81
      1951273.18     13879918.88       1950428.6     13881373.51
      1952098.82     13882298.13      1953122.71     13884069.19
      1955269.07     13883677.25        1956925.     13885167.44
       1958778.3     13884333.08      1959183.14     13886331.06
      1960626.47     13887221.46      1963078.22     13887966.72
      1964509.73     13886375.37        1966725.       13887875.

Type RM Length L Ch R = 1 ,81743   ,444,444,444
BEGIN DESCRIPTION:
Verde Creek 151.0
END DESCRIPTION:
XS GIS Cut Line= 3
      1912575.02     13865674.97        1912775.       13865275.
      1912875.01     13865074.98
#Sta/Elev= 30
  4552.6 1899.96  4587.1 1894.34  4630.3 1878.82  4641.4 1875.79  4660.9 1867.08
  4677.3 1858.67    4684 1853.78  4710.8 1841.15  4728.6 1834.36  4755.5 1827.95
    4798  1825.8  4842.7 1825.61  4885.3 1822.07  4925.5 1823.09    4997 1821.48
  5003.5 1820.55  5003.9 1820.05  5008.6 1820.55  5026.1 1820.99  5049.9 1826.97
  5069.7 1828.63    5088 1831.75  5102.3 1836.97  5130.1 1851.46  5140.2 1857.36
  5150.2 1865.09  5153.6 1868.68  5163.6 1875.11  5190.5 1883.75  5223.4 1888.93
#Mann= 3 ,-1 , 0
  4552.6      .1       0  5003.5     .05       0  5008.6      .1       0
Bank Sta=5003.5,5008.6
XS Rating Curve= 0 ,0
Exp/Cntr=0.3,0.1

Type RM Length L Ch R = 1 ,81299   ,473,473,473
BEGIN DESCRIPTION:
Verde Creek 150.0
END DESCRIPTION:
XS GIS Cut Line= 3
        1912925.     13865925.01        1913125.       13865525.
      1913175.01     13865274.97
#Sta/Elev= 30
  4552.5 1931.13  4566.2 1924.62  4619.9 1904.78  4636.6 1897.09  4653.4 1891.92
  4660.1 1887.89  4683.6 1879.23  4713.8 1865.47  4747.3 1853.15  4757.4  1847.1
  4758.9  1875.3  4762.2 1844.51  4765.6 1843.68  4799.1 1825.92  4822.6 1817.78
  4836.7 1816.16  4859.5 1815.82  4908.3 1817.82  4953.4 1816.85  4968.6 1818.38
  4982.1 1817.34  4994.5 1813.92  4994.9 1813.42  4999.6 1813.92  5040.1 1821.38
  5122.7 1822.69  5147.2 1829.65  5220.6 1863.75    5242 1869.85  5254.7 1872.04
#Mann= 3 ,-1 , 0
  4552.5      .1       0  4994.5     .05       0  4999.6      .1       0
Bank Sta=4994.5,4999.6
XS Rating Curve= 0 ,0
Exp/Cntr=0.3,0.1

Type RM Length L Ch R = 1 ,80826   ,470,470,470
BEGIN DESCRIPTION:
Verde Creek 149.0
END DESCRIPTION:
XS GIS Cut Line= 3
      1913824.99     13865874.99        1913475.       13865475.
      1913324.99     13865274.99
#Sta/Elev= 30
  4473.5 1941.95  4494.3 1940.34  4515.6 1934.23  4543.2 1921.48  4594.7 1903.33
  4650.5 1878.41  4652.3 1876.74  4660.3 1874.63  4699.4 1858.12  4756.8 1831.43
  4782.3 1822.31    4808 1818.21    4890 1814.48  4918.4 1809.58  4960.9 1809.82
  4975.3 1807.66  4975.7 1807.16  4980.5 1807.66  4984.3 1809.56  4991.1 1810.35
  5016.3 1809.65  5040.7 1810.95  5058.8 1815.69  5089.2 1816.98  5115.7 1820.81
  5155.6 1832.48  5194.2 1846.92  5215.6  1856.9  5230.6  1860.9    5255 1863.82
#Mann= 3 ,-1 , 0
  4473.5      .1       0  4975.3     .05       0  4980.5      .1       0
Bank Sta=4975.3,4980.5
XS Rating Curve= 0 ,0
Exp/Cntr=0.3,0.1

Type RM Length L Ch R = 1 ,80356   ,450,450,450
BEGIN DESCRIPTION:
Verde Creek 148.0
END DESCRIPTION:
XS GIS Cut Line= 3
      1914124.97     13865424.98        1913775.       13865125.
      1913474.97     13865024.99
#Sta/Elev= 30
  4543.7 1890.68    4569 1889.39  4597.4 1884.32  4620.4 1877.58  4648.1 1872.51
  4662.9 1866.42  4686.8 1845.88    4709 1833.27  4745.8 1816.12  4762.6 1811.62
  4798.2 1809.77  4852.8  1810.5  4873.3 1808.16  4891.1 1804.59  4912.8 1803.59
  4957.2 1804.26  4986.3 1802.25  4986.7 1801.75  4991.5 1802.25  5019.7 1806.78
    5044 1807.81  5060.6 1806.56  5079.8 1806.09  5095.6  1807.6    5124 1813.94
  5193.9 1832.75  5207.7  1837.9  5274.1 1857.83    5312 1863.91  5320.9  1864.1
#Mann= 5 ,-1 , 0
  4543.7      .1       0  4957.2     .07       0  4986.3     .05       0
  4991.5     .07       0  5060.6      .1       0
Bank Sta=4986.3,4991.5
XS Rating Curve= 0 ,0
Exp/Cntr=0.3,0.1

Type RM Length L Ch R = 1 ,79906   ,419,419,419
BEGIN DESCRIPTION:
Verde Creek 147.0
END DESCRIPTION:
XS GIS Cut Line= 3
      1914274.99     13865024.99        1914125.       13864875.
      1913825.01     13864475.02
#Sta/Elev= 30
  4792.7 1867.47  4820.1  1865.1  4822.3 1862.73  4828.4 1861.09    4835 1848.76
  4841.6 1841.71  4870.8 1823.22  4904.8 1807.41  4928.3  1801.2  4955.9 1798.92
  4966.5 1793.94  4980.8 1791.74  4981.2 1791.24  4986.2 1791.74  4994.3 1792.23
    5018 1800.48  5034.7 1801.47  5056.1 1805.99  5066.6 1806.15  5118.3 1804.21
  5131.1 1806.82  5165.4 1805.15  5229.7  1807.3  5258.4 1809.82  5351.9  1811.1
  5375.4 1813.67  5396.8 1820.26  5434.3 1836.95    5483 1864.01  5504.8 1868.87
#Mann= 5 ,-1 , 0
  4792.7      .1       0  4980.8     .05       0  4986.2      .1       0
  5066.6     .07       0  5258.4      .1       0
Bank Sta=4980.8,4986.2
XS Rating Curve= 0 ,0
Exp/Cntr=0.3,0.1

Type RM Length L Ch R = 1 ,79487   ,441,441,441
BEGIN DESCRIPTION:
Verde Creek 146.0
END DESCRIPTION:
XS GIS Cut Line= 3
      1914574.98     13864824.98        1914475.       13864675.
      1914075.02     13864275.02
#Sta/Elev= 30
  4815.1 1866.14  4832.6 1864.86  4843.8 1861.98  4854.2 1856.02    4866 1847.24
  4878.4 1840.23  4910.9 1824.23  4917.3  1820.3  4936.8 1811.38  4962.4 1803.95
  4968.8 1800.73  4979.6 1797.17  4987.6 1792.53    5010 1791.19  5010.4 1790.69
  5015.4 1791.19  5033.4  1793.6  5065.2 1793.21  5084.3 1794.09  5105.5  1797.8
  5135.2 1798.99  5168.7 1802.19  5207.1 1802.58  5305.4 1801.68  5345.2 1803.16
    5388 1806.24  5512.8 1813.78  5537.8 1819.64  5555.3 1824.91    5561  1827.4
#Mann= 5 ,-1 , 0
  4815.1      .1       0    5010     .05       0  5015.4      .1       0
  5207.1     .07       0    5388      .1       0
Bank Sta=5010,5015.4
XS Rating Curve= 0 ,0
Exp/Cntr=0.3,0.1

Type RM Length L Ch R = 1 ,79046   ,672,672,672
BEGIN DESCRIPTION:
Verde Creek 145.0
END DESCRIPTION:
XS GIS Cut Line= 3
        1914775.     13864574.98        1914725.       13864325.
      1914525.02     13863925.04
#Sta/Elev= 30
  4749.5 1832.09  4768.9 1830.68    4802 1825.04  4818.4 1815.22  4833.7 1807.83
  4858.1 1799.47  4870.9 1797.06  4906.6 1795.51  4931.6 1788.79  4986.7 1790.63
  5022.4 1787.52  5022.9 1787.02  5027.9 1787.52  5034.1 1789.13  5063.9 1789.99
    5093 1793.53  5106.4 1792.64    5207 1797.02  5229.8 1799.46  5246.6 1802.92
  5273.4 1811.59  5303.6 1825.91  5347.2 1850.08  5356.9 1857.31  5360.6 1861.54
  5365.8 1863.76  5387.4 1878.23  5397.1 1882.65  5432.9 1890.82  5451.6 1892.79
#Mann= 3 ,-1 , 0
  4749.5      .1       0  5022.4     .05       0  5027.9      .1       0
Bank Sta=5022.4,5027.9
XS Rating Curve= 0 ,0
Exp/Cntr=0.3,0.1

Type RM Length L Ch R = 1 ,78374   ,674,674,674
BEGIN DESCRIPTION:
Verde Creek 144.0
END DESCRIPTION:
XS GIS Cut Line= 3
        1914975.     13864675.01      1915195.47     13863927.52
      1914802.27     13863509.53
#Sta/Elev= 30
  4168.9 1844.06    4206 1837.34  4328.6 1823.09  4359.3 1813.19  4390.7 1806.23
  4409.3 1803.06  4424.9 1802.75  4496.9  1795.4  4556.2 1792.81  4754.8 1790.16
  4797.2 1787.33  4809.7 1786.13  4847.2 1786.73  4898.8 1785.42  4937.9 1784.84
  4970.8 1781.43  4971.2 1780.93  4976.4 1781.43  5012.1 1786.02  5056.3 1795.74
    5085 1804.88  5161.2 1846.19  5175.2 1856.08  5177.6 1859.97  5179.4 1861.28
  5202.3 1869.84  5243.5 1875.38  5323.7 1879.94  5359.8 1884.26  5522.1 1894.79
#Mann= 8 ,-1 , 0
  4168.9      .1       0  4390.7    .035       0  4556.2     .07       0
  4797.2      .1       0  4898.8    .035       0  4970.8    .035       0
  4976.4    .035       0  5012.1      .1       0
Bank Sta=4970.8,4976.4
XS Rating Curve= 0 ,0
Exp/Cntr=0.3,0.1

Type RM Length L Ch R = 1 ,77700   ,416,416,416
BEGIN DESCRIPTION:
Verde Creek 143.0
END DESCRIPTION:
XS GIS Cut Line= 3
      1915074.99     13864825.01        1915675.       13864125.
        1915975.       13864075.
#Sta/Elev= 30
  4077.7 1860.88  4092.9 1860.72  4126.2 1856.98  4215.4 1834.18  4252.5 1829.46
  4292.1 1821.74  4337.9 1802.01  4353.9 1801.33  4376.9 1796.28  4415.1 1791.56
  4421.8  1790.8  4520.8 1786.78  4618.5 1785.01  4810.3 1785.31  4883.2 1779.81
  4919.6 1779.59  4985.8 1777.37  4986.3 1776.87  4994.2 1777.37  5014.6 1779.13
  5032.9 1782.93  5108.9 1787.47  5142.3 1793.55  5160.6 1799.88  5181.9 1809.95
  5245.8 1846.55  5257.9 1855.29    5261 1859.45    5264 1860.78  5303.8 1861.17
#Mann= 7 ,-1 , 0
  4077.7      .1       0  4415.1     .07       0  4421.8    .035       0
  4520.8     .07       0  4919.6      .1       0  4985.8     .05       0
  4994.2      .1       0
Bank Sta=4985.8,4994.2
XS Rating Curve= 0 ,0
Exp/Cntr=0.3,0.1

Type RM Length L Ch R = 1 ,77284   ,439,439,439
BEGIN DESCRIPTION:
Verde Creek 142.0
END DESCRIPTION:
XS GIS Cut Line= 3
      1915425.02     13864874.98        1915825.       13864475.
      1915975.02     13864174.97
#Sta/Elev= 30
  4434.8 1798.91  4445.5 1798.87    4524 1790.64    4579 1786.78  4648.8 1782.54
  4732.8 1780.79  4848.7  1781.3  4860.7 1780.56    4877 1776.56  4885.5  1775.9
  4919.5 1776.01  4932.2 1779.04  4939.2 1779.25  4987.3 1775.81  4987.8 1775.31
  4995.8 1775.81  5051.4 1776.01    5067 1780.66    5155 1782.99  5178.9 1786.52
  5205.7 1796.56  5225.8 1806.31  5239.2 1815.23  5252.6 1822.21  5259.4 1827.03
  5286.2  1842.6  5299.6 1847.97    5303 1850.61  5316.4    1854  5335.9 1855.69
#Mann= 7 ,-1 , 0
  4434.8      .1       0    4524     .07       0    4579    .035       0
  4648.8     .07       0  4848.7      .1       0  4987.3     .05       0
  4995.8      .1       0
Bank Sta=4987.3,4995.8
XS Rating Curve= 0 ,0
Exp/Cntr=0.3,0.1

Type RM Length L Ch R = 1 ,76845   ,465,465,465
BEGIN DESCRIPTION:
Verde Creek 141.0
END DESCRIPTION:
XS GIS Cut Line= 3
      1915474.98     13865125.01        1915875.       13864825.
      1916274.98     13864675.01
#Sta/Elev= 30
  4499.9  1809.2  4532.1 1805.09  4539.6 1803.26  4580.8 1796.35  4603.3 1795.77
  4630.1  1792.5  4674.6  1789.1  4750.7 1785.62  4824.6 1780.59    4863 1780.43
    4908 1778.55  4929.6 1777.63  4937.1 1778.24  4948.3  1776.6  4961.6 1776.04
  5007.3 1775.84  5019.9 1775.83  5020.4 1775.33  5028.8 1775.83  5109.6  1776.5
  5112.9 1776.73  5128.9 1781.15  5166.1 1784.09    5225 1784.04  5267.8 1785.48
  5326.4 1788.05    5359 1795.66  5378.8  1800.3  5391.6 1804.88  5427.1 1815.34
#Mann= 10 ,-1 , 0
  4499.9      .1       0  4630.1     .07       0  4750.7    .035       0
    4908     .07       0  5007.3    .033       0  5019.9     .05       0
  5028.8    .033       0  5166.1      .1       0  5267.8     .07       0
    5359      .1       0
Bank Sta=5019.9,5028.8
XS Rating Curve= 0 ,0
Exp/Cntr=0.3,0.1

Type RM Length L Ch R = 1 ,76380   ,473,473,473
BEGIN DESCRIPTION:
Verde Creek 140.0
END DESCRIPTION:
XS GIS Cut Line= 3
        1915575.       13865475.        1915975.       13865225.
      1916375.01     13864824.99
#Sta/Elev= 30
  4528.3 1855.98  4553.9 1852.23  4578.7 1842.65    4606 1834.04  4621.8  1827.4
  4638.8 1822.67  4670.7 1808.14  4684.8 1802.98  4710.7 1798.57  4741.4 1792.02
  4757.7 1789.72  4780.3 1784.78  4794.5 1784.87  4815.2 1782.04  4872.5  1778.9
  4904.2 1777.53  4918.3 1775.97  4991.1 1775.92    5077 1775.73  5077.5 1775.23
  5085.9 1775.73  5160.9 1775.87  5233.5 1778.18  5326.3 1779.02  5445.1 1783.79
  5467.5 1786.44  5494.3 1794.86  5535.4  1810.7  5556.6 1820.88  5565.7 1823.76
#Mann= 8 ,-1 , 0
  4528.3     .07       0    4606      .1       0  4872.5    .035       0
  4991.1    .033       0    5077    .033       0  5085.9    .033       0
  5233.5     .07       0  5494.3      .1       0
Bank Sta=5077,5085.9
XS Rating Curve= 0 ,0
Exp/Cntr=0.3,0.1

Type RM Length L Ch R = 1 ,75907   ,459,459,459
BEGIN DESCRIPTION:
Verde Creek 139.0
END DESCRIPTION:
XS GIS Cut Line= 3
      1915774.96     13865725.01        1916175.       13865625.
      1916574.97     13865225.03
#Sta/Elev= 30
  4583.1 1820.65  4637.5 1803.51  4649.9 1800.67  4665.3  1795.3  4705.5 1785.77
  4711.7 1784.95  4758.1 1783.58  4767.3 1782.52  4779.9 1782.92  4797.4 1781.95
  4831.6 1781.58  4858.2 1783.66  4912.7 1783.78  4962.2 1781.11  4967.7 1780.14
  4974.6  1776.6  4977.7 1775.81  5008.9  1775.7  5009.4  1775.2    5018  1775.7
  5105.7    1776  5362.5  1775.8  5375.3 1776.64  5392.2 1779.53  5412.3    1779
  5438.3 1779.72  5463.2 1781.74  5505.6 1788.88  5518.3 1791.53  5561.1 1802.96
#Mann= 6 ,-1 , 0
  4583.1      .1       0  4797.4     .07       0  5008.9     .05       0
    5018     .07       0  5105.7    .033       0  5438.3      .1       0
Bank Sta=5008.9,5018
XS Rating Curve= 0 ,0
Exp/Cntr=0.3,0.1

Type RM Length L Ch R = 1 ,75448   ,423,423,423
BEGIN DESCRIPTION:
Verde Creek 138.0
END DESCRIPTION:
XS GIS Cut Line= 3
      1915925.02     13866374.98        1916325.       13866025.
      1917024.96     13865575.03
#Sta/Elev= 30
  4468.3 1866.52  4502.7 1862.17  4550.7  1853.5  4582.5 1842.65  4626.3 1830.11
  4662.1 1822.42    4694 1812.08  4733.9 1803.27  4869.4 1783.65  4903.4 1781.85
  4960.6 1777.54  4976.4 1776.02  4976.9 1775.52  4985.7 1776.02  5045.2 1776.24
  5534.7    1778  5535.7 1823.43  5537.1 1883.48  5542.7 1778.24  5621.2 1777.08
  5635.5 1784.38  5648.1  1786.2  5692.5 1802.98  5721.1 1818.39  5742.4 1833.09
  5756.7 1840.84  5772.8 1867.91  5778.1 1872.56  5783.6 1874.77  5831.9 1878.42
#Mann= 7 ,-1 , 0
  4468.3     .07       0  4903.4    .035       0  4960.6     .07       0
  4976.4     .05       0  4985.7     .07       0  5045.2    .033       0
  5783.6      .1       0
Bank Sta=4976.4,4985.7
XS Rating Curve= 0 ,0
Exp/Cntr=0.3,0.1

Type RM Length L Ch R = 1 ,75025   ,413,413,413
BEGIN DESCRIPTION:
Verde Creek 137.0
END DESCRIPTION:
XS GIS Cut Line= 3
      1916174.97     13866675.03        1916525.       13866375.
      1917125.02     13865674.98
#Sta/Elev= 30
    4539 1868.52  4576.3 1864.09  4599.4 1855.65  4636.2 1838.68  4706.2 1814.32
  4779.1 1797.33  4821.7 1790.79  4824.8 1790.13  4836.6 1787.22  4871.3  1784.9
  4895.8 1781.31  4945.1 1779.74  4974.9 1776.27    5081 1776.31  5403.4 1776.93
  5450.4  1775.7  5450.9  1775.2  5459.8  1775.7  5699.7 1776.61  5711.6 1779.86
  5739.2 1780.91    5755 1790.17  5766.9 1799.43  5794.5 1824.38  5818.9 1841.19
  5832.7 1848.99  5843.7 1867.79  5851.6 1872.75  5877.4 1876.06    5922  1878.5
#Mann= 7 ,-1 , 0
    4539     .07       0  4821.7    .035       0  4824.8     .07       0
    5081    .033       0  5450.4     .05       0  5459.8    .033       0
  5877.4      .1       0
Bank Sta=5450.4,5459.8
XS Rating Curve= 0 ,0
Exp/Cntr=0.3,0.1

Type RM Length L Ch R = 1 ,74612   ,212,212,212
BEGIN DESCRIPTION:
Verde Creek 136.0
END DESCRIPTION:
XS GIS Cut Line= 3
        1916267.     13866960.81      1916723.55     13866659.67
      1917501.79     13866156.43
#Sta/Elev= 30
  4463.2 1878.96  4526.6 1872.35  4573.3 1864.96    4602 1855.37  4617.7 1848.24
  4628.6 1840.64  4704.9 1810.82  4740.6  1800.3  4756.6 1797.31  4767.3    1793
  4792.5 1791.07  4810.5 1784.13  4835.6 1784.08    4852 1778.63  4885.9 1775.84
  4961.7 1775.72  4962.2 1775.22  4971.1 1775.72  4974.1 1775.85  4993.7  1775.8
  5740.5 1776.45  5754.8 1781.06  5776.2  1782.8  5813.8 1801.21  5833.7 1814.11
  5836.3 1815.64  5849.8 1825.34  5883.4 1836.03    5905 1840.82  5936.9  1845.1
#Mann= 8 ,-1 , 0
  4463.2     .07       0  4792.5    .035       0  4961.7    .033       0
  4971.1    .035       0  4974.1     .07       0  4993.7    .033       0
  5833.7     .07       0  5836.3      .1       0
Bank Sta=4961.7,4971.1
XS Rating Curve= 0 ,0
Exp/Cntr=0.3,0.1

Type RM Length L Ch R = 1 ,74400   ,212,212,212
BEGIN DESCRIPTION:
Verde Creek D5
END DESCRIPTION:
XS GIS Cut Line= 6
      1916292.47      13867121.1      1916804.63     13866795.58
      1916926.16     13866730.47      1917299.42     13866565.54
      1917442.65     13866526.48      1917991.95     13866401.05
#Sta/Elev= 30
    4488 1884.44  4573.7 1879.16  4727.2 1865.29  4733.2 1863.27  4754.3 1838.03
  4769.6 1824.68    4806 1801.37  4827.2  1793.5  4869.3 1790.57  4915.2 1775.25
  5103.8 1777.15    5136 1782.74  5175.7 1786.96  5229.2 1782.82  5235.4 1786.57
    5282 1782.33  5291.3 1785.84  5357.4 1783.16  5362.9 1786.35    5646 1787.23
  5749.1 1787.65    5793 1786.11  5832.7 1777.98  6002.4  1774.5  6002.9    1774
  6011.8  1774.5  6027.6 1784.93  6123.4 1807.14    6263 1848.83  6352.7 1859.85
#Mann= 11 ,-1 , 0
    4488      .1       0  4573.7     .07       0  4869.3    .035       0
    5136     .07       0  5175.7    .035       0  5291.3     .07       0
    5646    .035       0  5749.1     .07       0  6002.4    .035       0
  6011.8     .07       0  6123.4      .1       0
Bank Sta=6002.4,6011.8
XS Rating Curve= 0 ,0
Exp/Cntr=0.3,0.1

Type RM Length L Ch R = 1 ,74188   ,438,438,438
BEGIN DESCRIPTION:
Verde Creek 135.0
END DESCRIPTION:
XS GIS Cut Line= 3
      1916575.01     13867174.99        1916825.       13867025.
      1918019.96     13866549.02
#Sta/Elev= 30
  4713.1 1867.77  4731.1 1866.29    4737 1865.71  4758.4 1862.09  4768.9 1848.26
  4821.4  1810.7  4878.3 1777.95  4886.6 1772.27  4905.4 1770.25  4922.9 1762.83
  4947.4 1761.44  5077.7 1760.15  5126.1 1764.61  5174.6 1756.34  5539.5    1760
    5575 1758.77  5612.4  1752.1  5618.8 1751.21  5625.2 1751.12  5625.7 1750.62
  5634.6 1751.12  5736.5 1759.77  5778.5 1771.69  5828.5 1769.82  5952.8 1772.54
  6001.3 1780.93  6103.1 1806.08  6224.1 1848.45  6254.9  1856.3  6290.9 1860.51
#Mann= 10 ,-1 , 0
  4713.1      .1       0  4731.1     .07       0    4737      .1       0
  4878.3    .035       0  5612.4     .07       0  5618.8      .1       0
  5625.2    .035       0  5634.6      .1       0  5828.5     .07       0
  6103.1      .1       0
Bank Sta=5625.2,5634.6
XS Rating Curve= 0 ,0
Exp/Cntr=0.3,0.1

Type RM Length L Ch R = 1 ,73750   ,370,370,370
BEGIN DESCRIPTION:
Verde Creek 134.0
END DESCRIPTION:
XS GIS Cut Line= 3
      1916725.01       13867225.        1917125.       13867325.
      1918013.13     13867431.57
#Sta/Elev= 30
  4595.5 1809.25  4620.1 1795.34  4671.1 1772.16  4697.4 1762.84  4709.8 1760.51
    4716 1757.26  4814.4 1754.06  4836.6    1756  4873.7 1752.22  5007.8 1750.42
  5163.5 1754.46  5177.4 1753.41    5197 1746.82  5197.5 1746.32  5206.5 1746.82
    5336 1749.65  5363.2 1758.97  5372.3 1760.56  5398.7 1758.92  5456.9 1765.45
  5482.3  1765.3  5495.8 1769.09  5574.7 1776.94  5595.9 1782.49  5668.4 1794.65
  5722.8 1806.25  5795.3 1831.56  5852.7 1855.22  5876.9 1862.36  5902.3 1866.92
#Mann= 5 ,-1 , 0
  4595.5      .1       0  4814.4    .035       0  5163.5      .1       0
    5197    .035       0  5206.5      .1       0
Bank Sta=5197,5206.5
XS Rating Curve= 0 ,0
Exp/Cntr=0.3,0.1

Type RM Length L Ch R = 1 ,73380   ,460,460,460
BEGIN DESCRIPTION:
Verde Creek 133.0
END DESCRIPTION:
XS GIS Cut Line= 3
      1916574.97     13867274.97      1916984.99     13867637.15
      1917517.27       13867801.
#Sta/Elev= 30
  4503.9 1867.62  4539.8  1863.2  4571.8 1852.93  4583.9 1845.46  4667.3 1806.21
  4707.5 1793.52  4739.2 1781.12    4756 1770.59  4770.9 1756.79  4786.1 1748.39
  4794.9 1745.07  4807.6 1743.75    4848 1746.04  4872.1 1743.19  4880.1  1744.6
  4901.9 1742.69  4952.4 1742.27  4979.4 1742.19  4991.9 1740.19  4992.4 1739.69
  5001.6 1740.19  5013.8    1742  5037.4 1749.71  5047.3 1751.68  5246.8 1753.33
  5297.7 1755.51  5328.1 1758.57    5429 1761.76  5558.6 1772.57  5607.9 1776.74
#Mann= 8 ,-1 , 0
  4503.9      .1       0  4786.1     .07       0  4901.9      .1       0
  4952.4     .07       0  4991.9     .05       0  5001.6     .07       0
  5037.4    .035       0  5558.6      .1       0
Bank Sta=4991.9,5001.6
XS Rating Curve= 0 ,0
Exp/Cntr=0.3,0.1

Type RM Length L Ch R = 1 ,72920   ,512,512,512
BEGIN DESCRIPTION:
Verde Creek 132.0
END DESCRIPTION:
XS GIS Cut Line= 3
      1916475.03     13867675.03      1916635.66     13867814.86
      1917475.25       13867884.
#Sta/Elev= 30
  4694.2 1870.77  4736.4 1863.93    4747 1858.73  4751.3 1854.77  4764.1  1847.1
  4808.7 1824.86  4856.7 1798.16  4945.5 1757.42  4970.3 1741.48  4997.9 1737.29
  4998.4 1736.79  5007.6 1737.29  5043.4 1740.58  5114.1 1746.04    5142 1744.63
  5277.5 1747.81  5318.8 1748.55  5381.9 1752.42  5403.1 1752.14  5436.2 1755.53
  5460.3 1754.66  5481.3 1758.04  5511.4 1757.81  5536.5 1760.14  5544.5 1761.31
  5583.7  1761.9  5629.4 1766.99  5661.9 1767.28  5700.8 1772.24  5749.6 1775.58
#Mann= 8 ,-1 , 0
  4694.2      .1       0  4997.9     .05       0  5007.6      .1       0
  5043.4     .07       0    5142      .1       0  5277.5    .035       0
  5536.5     .07       0  5700.8      .1       0
Bank Sta=4997.9,5007.6
XS Rating Curve= 0 ,0
Exp/Cntr=0.3,0.1

Type RM Length L Ch R = 1 ,72408   ,453,453,453
BEGIN DESCRIPTION:
Verde Creek 131.0
END DESCRIPTION:
XS GIS Cut Line= 4
      1916274.95     13868074.99      1916893.69     13868224.39
        1917025.       13868225.      1917512.53     13868240.43
#Sta/Elev= 30
  4236.8 1839.77  4262.2 1835.24    4297 1824.36  4309.5 1819.53  4324.4 1811.63
  4433.7 1770.51    4476 1754.48  4498.4 1753.73  4513.3 1751.32  4690.4 1747.94
  4897.6 1746.67  4923.5 1746.52  4966.4 1736.16  4999.6 1735.17  5000.1 1734.67
  5009.4 1735.17  5052.5 1739.38  5100.6 1749.86  5113.7 1750.53  5130.6 1752.99
  5181.6 1765.08  5210.4 1769.96  5272.9 1777.77  5329.4 1788.12  5370.7 1794.08
  5427.1 1803.59  5436.7 1806.17  5448.7 1806.18  5482.9 1813.78  5492.4 1816.66
#Mann= 9 ,-1 , 0
  4236.8      .1       0  4433.7     .07       0  4897.6      .1       0
  4999.6     .05       0  5009.4      .1       0  5113.7    .035       0
  5210.4      .1       0  5329.4     .07       0  5482.9      .1       0
Bank Sta=4999.6,5009.4
XS Rating Curve= 0 ,0
Exp/Cntr=0.3,0.1

Type RM Length L Ch R = 1 ,71955   ,488,488,488
BEGIN DESCRIPTION:
Verde Creek 130.0
END DESCRIPTION:
XS GIS Cut Line= 3
      1916316.81     13868287.22        1917175.       13868625.
      1917575.01       13868425.
#Sta/Elev= 30
  4076.8 1772.16  4089.8 1769.63  4112.9 1759.96    4122 1756.64  4140.5 1756.14
  4163.9  1752.4  4237.7 1749.98    4750 1742.46  4763.6 1742.56  4831.3 1734.13
  4847.4 1735.68  4863.5 1733.84  4902.2  1736.2  4945.6 1736.02  4989.3 1733.11
  5000.1 1730.32  5000.6 1729.82  5009.9 1730.32  5019.1 1737.19  5032.5 1741.91
  5116.3 1745.09  5183.3 1751.48  5210.3 1755.29  5231.7 1761.71  5295.3 1787.99
  5334.4 1805.93  5361.2 1820.75  5404.8 1842.35  5431.6 1853.73  5446.3 1856.28
#Mann= 7 ,-1 , 0
  4076.8    .035       0  4112.9     .07       0    4750      .1       0
  5000.1     .05       0  5009.9      .1       0  5183.3     .07       0
  5295.3      .1       0
Bank Sta=5000.1,5009.9
XS Rating Curve= 0 ,0
Exp/Cntr=0.3,0.1

Type RM Length L Ch R = 1 ,71467   ,444,444,444
BEGIN DESCRIPTION:
Verde Creek 129.0
END DESCRIPTION:
XS GIS Cut Line= 3
      1916178.76     13869049.33        1917075.       13869075.
        1917475.       13869375.
#Sta/Elev= 30
  4107.9  1756.5    4156 1756.51    4220  1753.8  4370.5 1750.29  4648.2 1743.67
  4676.4 1741.55  4801.3 1737.04  4858.2 1733.46  4894.3 1730.93    4938 1731.72
  4981.8 1726.92  4982.3 1726.42  4993.5 1726.92  4996.4 1732.72  5002.4 1739.34
  5009.4 1740.52  5066.4 1738.63  5137.3 1738.04  5225.7 1738.52  5249.4 1740.09
  5275.6 1744.09  5292.1 1749.47  5316.9 1760.11  5399.4 1804.07  5459.4 1841.04
  5470.6 1850.22  5476.4 1860.27  5485.6 1869.91  5496.9 1875.28  5504.5 1876.85
#Mann= 9 ,-1 , 0
  4107.9     .07       0    4220    .035       0  4370.5     .07       0
  4676.4    .035       0  4858.2      .1       0  4981.8     .05       0
  4993.5      .1       0  5066.4     .07       0  5137.3      .1       0
Bank Sta=4981.8,4993.5
XS Rating Curve= 0 ,0
Exp/Cntr=0.3,0.1

Type RM Length L Ch R = 1 ,71023   ,448,448,448
BEGIN DESCRIPTION:
Verde Creek 128.0
END DESCRIPTION:
XS GIS Cut Line= 3
      1916176.09     13869595.39        1917025.       13869475.
      1917424.98       13869425.
#Sta/Elev= 30
  4142.6 1774.12  4172.7 1772.33  4245.4 1761.92  4263.6 1758.17  4281.8 1757.64
  4289.3 1755.55  4329.6 1750.15  4358.8 1750.95    4409 1746.48  4589.3 1739.77
  4789.2 1736.22  4839.3 1734.45  4889.2 1728.29  4936.3 1728.34  4969.6 1725.27
  4969.8 1724.35  4970.3 1723.85  4981.5 1724.35  4993.8  1725.2  5005.9 1731.81
    5012 1733.61    5033 1735.72  5120.8 1734.29  5193.4 1736.36  5202.5  1738.2
  5229.7 1751.02    5278 1781.58  5312.9 1798.09  5335.5 1806.55  5403.1 1840.43
#Mann= 7 ,-1 , 0
  4142.6     .07       0  4289.3    .035       0  4589.3     .07       0
  4789.2    .035       0  4889.2      .1       0  4969.8     .05       0
  4981.5      .1       0
Bank Sta=4969.8,4981.5
XS Rating Curve= 0 ,0
Exp/Cntr=0.3,0.1

Type RM Length L Ch R = 1 ,70575   ,447,447,447
BEGIN DESCRIPTION:
Verde Creek 127.0
END DESCRIPTION:
XS GIS Cut Line= 3
      1916550.03     13870225.64        1917225.       13869825.
        1917575.       13869475.
#Sta/Elev= 30
  4220.8 1758.11  4333.4 1748.62  4392.3 1748.17  4519.9 1743.17  4626.5 1740.39
  4640.4 1738.57  4722.4 1737.85    4786 1735.09  4859.6 1732.93  4881.2 1731.24
  4894.5 1726.79  4912.6 1724.09  4964.9 1724.19  4986.8 1721.27  4987.3 1720.77
  4998.8 1721.27  5031.5 1722.27  5052.7 1725.79  5091.8 1729.02  5125.3 1728.45
  5201.2 1734.13  5250.5 1746.16  5288.7 1763.06  5383.7 1820.04  5428.7 1851.47
  5439.7 1866.14  5447.3 1870.79  5454.1 1877.13    5460 1879.03  5500.7 1882.14
#Mann= 8 ,-1 , 0
  4220.8      .1       0  4392.3     .05       0  4519.9     .07       0
  4722.4     .05       0    4786     .07       0  4859.6      .1       0
  4986.8     .05       0  4998.8      .1       0
Bank Sta=4986.8,4998.8
XS Rating Curve= 0 ,0
Exp/Cntr=0.3,0.1

Type RM Length L Ch R = 1 ,70128   ,456,456,456
BEGIN DESCRIPTION:
Verde Creek 126.0
END DESCRIPTION:
XS GIS Cut Line= 3
      1917124.97     13870425.03        1917525.       13870125.
      1917875.03     13869724.96
#Sta/Elev= 30
  4504.3 1739.32  4549.8 1737.78  4589.9 1732.82  4631.3 1729.53  4724.2 1725.53
  4807.9 1724.42  4828.6 1724.22  4851.7 1724.49  4869.8 1721.93  4945.5 1719.88
  4971.7 1718.49  4976.9 1716.92  4977.4 1716.42  4989.1 1716.92  5024.6 1720.12
  5036.6 1723.97  5049.8 1730.12  5060.4 1732.05  5168.1  1729.5  5227.1  1730.3
  5267.8 1731.09  5303.6 1733.47  5317.7 1736.12  5331.6  1737.2  5367.3 1744.61
  5392.9 1751.84  5407.3 1757.51  5455.1 1780.03    5503 1801.06  5535.9 1810.78
#Mann= 9 ,-1 , 0
  4504.3      .1       0  4589.9     .05       0  4631.3      .1       0
  4807.9     .05       0  4828.6      .1       0  4976.9     .05       0
  4989.1      .1       0  5227.1     .07       0  5367.3      .1       0
Bank Sta=4976.9,4989.1
XS Rating Curve= 0 ,0
Exp/Cntr=0.3,0.1

Type RM Length L Ch R = 1 ,69672   ,485,485,485
BEGIN DESCRIPTION:
Verde Creek 125.0
END DESCRIPTION:
XS GIS Cut Line= 3
      1917430.42     13870984.08        1917725.       13870525.
      1917939.01      13869790.4
#Sta/Elev= 30
  4444.6 1753.03    4628  1745.4    4660  1743.1  4732.6 1741.13    4767 1739.48
  4784.8 1737.69  4854.7  1722.1  4884.1  1718.4  4955.9 1715.83  4961.7 1716.35
    5007    1713  5007.5  1712.5  5019.4    1713  5039.7 1716.74  5050.7 1721.45
  5060.1 1723.72  5096.6 1726.13    5168 1727.59    5371 1728.16  5472.6 1728.41
  5553.8 1728.53  5603.8 1729.89  5610.1 1730.76  5616.3  1733.3  5628.8 1734.22
  5635.1 1735.81  5641.3  1739.3  5650.7 1742.52  5695.7 1755.79  5755.2 1771.03
#Mann= 10 ,-1 , 0
  4444.6    .035       0  4732.6     .07       0  4884.1     .05       0
  4961.7      .1       0    5007     .05       0  5019.4      .1       0
    5168     .07       0    5371      .1       0  5472.6     .07       0
  5695.7      .1       0
Bank Sta=5007,5019.4
XS Rating Curve= 0 ,0
Exp/Cntr=0.3,0.1

Type RM Length L Ch R = 1 ,69187   ,419,419,419
BEGIN DESCRIPTION:
Verde Creek 124.0
END DESCRIPTION:
XS GIS Cut Line= 3
      1918297.15      13870992.7        1918175.       13870425.
      1918056.36     13869721.63
#Sta/Elev= 30
  4419.6 1771.04  4421.5 1770.83  4531.7 1762.16  4577.1 1757.19  4598.6 1752.36
  4615.1 1752.62  4650.7 1748.36  4672.2 1748.05  4705.9 1745.17  4755.1 1739.45
  4819.5 1729.99  4958.8 1717.11  4979.6 1712.37  5006.5 1710.72    5007 1710.22
    5019 1710.72  5032.7 1712.22  5061.3 1711.65  5071.8 1713.08  5092.6 1713.31
    5104  1715.6  5126.4 1723.19  5144.7 1725.96  5196.6  1725.4  5498.7  1726.6
  5566.4 1728.18  5590.2 1732.38  5627.3 1738.01  5660.7 1745.86  5713.6 1764.56
#Mann= 7 ,-1 , 0
  4419.6     .07       0  4421.5    .035       0  4958.8      .1       0
  5006.5     .05       0    5019      .1       0  5196.6     .07       0
  5590.2      .1       0
Bank Sta=5006.5,5019
XS Rating Curve= 0 ,0
Exp/Cntr=0.3,0.1

Type RM Length L Ch R = 1 ,68768   ,443,443,443
BEGIN DESCRIPTION:
Verde Creek 123.0
END DESCRIPTION:
XS GIS Cut Line= 3
      1918524.99     13870474.96        1918475.       13870175.
      1918204.64     13869536.04
#Sta/Elev= 30
  4691.4 1734.72  4790.1 1725.97  4812.3 1720.44  4824.4 1715.69  4830.5  1714.6
  4919.9 1712.25  4946.1 1711.65  4969.7 1708.85  5001.5 1707.53    5002 1707.03
    5014 1707.53  5014.1 1708.29  5023.2 1709.73  5031.5 1716.29  5043.5 1722.13
  5057.6 1722.55  5064.4  1724.2  5105.6 1722.93  5187.9 1722.77  5433.3 1724.14
  5502.9 1726.06  5515.9 1727.78  5532.2 1731.81  5561.1 1742.84  5587.5  1754.3
  5590.8 1756.49  5597.3 1758.27  5606.9 1763.54  5622.9 1769.61  5689.3  1800.8
#Mann= 7 ,-1 , 0
  4691.4    .035       0  4790.1     .07       0  4919.9      .1       0
  5001.5     .05       0    5014      .1       0  5187.9     .07       0
  5433.3      .1       0
Bank Sta=5001.5,5014
XS Rating Curve= 0 ,0
Exp/Cntr=0.3,0.1

Type RM Length L Ch R = 1 ,68325   ,472,472,472
BEGIN DESCRIPTION:
Verde Creek 122.0
END DESCRIPTION:
XS GIS Cut Line= 3
      1919110.42     13870420.27        1918825.       13869925.
      1918796.55     13869027.48
#Sta/Elev= 30
  4428.6 1749.29  4456.3 1746.44    4496 1744.04  4502.5 1742.19  4540.6 1739.43
  4606.4 1735.19  4627.2 1735.74  4650.1 1733.83  4683.1 1733.43  4715.7 1730.34
  4790.9 1728.56  4945.6 1719.46  4953.2 1717.72  4963.6 1709.66  4970.4 1706.15
  4979.5 1705.21    4980 1704.71  4992.2 1705.21  5040.5 1707.42  5112.5 1706.58
  5137.8 1708.74  5187.6 1717.12  5199.6 1720.25  5226.6 1720.47  5513.6 1723.97
  5706.8 1728.76  5719.3 1731.34  5739.8 1734.75  5763.9    1741  5898.2 1786.91
#Mann= 8 ,-1 , 0
  4428.6     .07       0  4456.3      .1       0  4650.1     .07       0
  4945.6      .1       0  4979.5     .05       0  4992.2      .1       0
  5226.6     .07       0  5719.3      .1       0
Bank Sta=4979.5,4992.2
XS Rating Curve= 0 ,0
Exp/Cntr=0.3,0.1

Type RM Length L Ch R = 1 ,67853   ,444,444,444
BEGIN DESCRIPTION:
Verde Creek 121.0
END DESCRIPTION:
XS GIS Cut Line= 3
      1919245.33     13870308.25        1919175.       13869625.
        1919175.     13869024.96
#Sta/Elev= 30
  4308.1 1742.61    4413 1735.12  4499.2 1730.89  4591.6 1724.81  4669.8 1722.94
  4909.2 1712.13  4929.6 1710.28  4944.5 1703.19  5001.3 1700.52  5001.8 1700.02
  5014.2 1700.52  5025.7 1702.48  5058.7 1702.11  5088.7 1705.01  5106.3  1711.1
  5128.2 1715.56  5238.3 1716.28  5337.7 1726.19  5368.2 1740.66  5400.7 1761.02
  5415.7 1768.61  5436.7 1776.18  5463.7 1791.69  5487.7 1808.11  5499.7 1822.75
  5532.7 1848.51  5550.7 1860.68  5556.3 1868.15  5562.7 1872.84    5595 1874.19
#Mann= 6 ,-1 , 0
  4308.1      .1       0    4413    .035       0  4499.2     .07       0
  4909.2      .1       0  5001.3     .05       0  5014.2      .1       0
Bank Sta=5001.3,5014.2
XS Rating Curve= 0 ,0
Exp/Cntr=0.3,0.1

Type RM Length L Ch R = 1 ,67409   ,435,435,435
BEGIN DESCRIPTION:
Verde Creek 120.0
END DESCRIPTION:
XS GIS Cut Line= 3
        1919525.     13870174.95        1919575.       13869575.
      1919374.98     13869074.95
#Sta/Elev= 30
  4391.8  1735.3    4520 1725.35  4641.7 1718.98  4688.5 1715.41  4733.7 1714.43
  4881.4 1707.72  4900.5 1705.51  4926.4  1705.2  4950.4  1703.5  4989.6 1703.57
  5011.9 1699.28  5047.2 1698.62  5047.4 1698.62  5047.9 1698.12  5060.3 1698.62
  5063.6 1701.47  5097.2  1708.4  5173.3 1711.99  5189.5 1716.57  5219.5 1729.34
  5241.3    1740  5244.5 1740.41  5260.7  1748.8  5280.1  1753.6  5328.5 1774.27
  5380.2 1793.96  5396.4 1801.18  5506.2 1860.53  5517.2 1864.56  5532.4 1865.96
#Mann= 4 ,-1 , 0
  4391.8    .035       0  5047.2      .1       0  5047.4    .035       0
  5060.3      .1       0
Bank Sta=5047.4,5060.3
XS Rating Curve= 0 ,0
Exp/Cntr=0.3,0.1

Type RM Length L Ch R = 1 ,66974   ,432,432,432
BEGIN DESCRIPTION:
Verde Creek 119.0
END DESCRIPTION:
XS GIS Cut Line= 4
      1919724.99     13870275.03        1919975.       13869675.
      1919984.25     13869544.96      1919625.03     13869075.03
#Sta/Elev= 30
  4345.5 1741.48  4381.3 1739.01  4504.5 1729.44  4582.5  1718.9    4706 1710.74
  4878.2 1702.47    4914 1699.86    4953 1699.26  4962.4 1697.19  4962.9 1696.69
  4975.4 1697.19  4985.5 1698.34  5031.4 1698.63  5046.4 1701.28  5052.4 1704.87
  5064.1 1708.71  5073.5 1709.36  5143.7 1708.03  5209.7 1709.06  5260.4 1711.53
  5306.5 1715.03  5343.3 1718.97  5408.8 1729.38  5451.6 1738.63  5486.8 1749.73
  5501.9 1756.18  5515.8 1758.69  5524.3 1762.59  5592.5  1785.2  5717.4 1829.93
#Mann= 7 ,-1 , 0
  4345.5      .1       0  4381.3    .035       0  4878.2      .1       0
  4962.4     .05       0  4975.4      .1       0  5260.4     .07       0
  5306.5      .1       0
Bank Sta=4962.4,4975.4
XS Rating Curve= 0 ,0
Exp/Cntr=0.3,0.1

Type RM Length L Ch R = 1 ,66542   ,484,484,484
BEGIN DESCRIPTION:
Verde Creek 118.0
END DESCRIPTION:
XS GIS Cut Line= 3
      1920424.99     13869974.97        1920375.       13869775.
      1919925.02     13869175.02
#Sta/Elev= 30
  4793.9 1721.79  4827.1  1721.3  4852.4 1719.67  4859.3 1718.31  4867.8 1715.05
  4898.8 1698.75    4908 1696.14  4948.2  1694.5  4965.6 1695.14  4976.1 1694.24
  5017.2  1693.6  5017.7  1693.1  5030.4  1693.6  5036.7 1694.89  5049.7 1694.58
    5061 1700.24  5073.1 1704.79  5083.8 1705.95  5111.5 1706.09  5173.5 1705.21
  5349.5 1705.75  5448.1 1709.64  5484.5 1711.77  5507.4 1714.62  5548.5 1718.01
  5574.3 1721.49  5611.3 1727.91  5668.8 1737.96  5724.3 1750.43    5750 1757.08
#Mann= 6 ,-1 , 0
  4793.9      .1       0  5017.2     .05       0  5030.4      .1       0
  5111.5     .07       0  5507.4      .1       0  5611.3     .07       0
Bank Sta=5017.2,5030.4
XS Rating Curve= 0 ,0
Exp/Cntr=0.3,0.1

Type RM Length L Ch R = 1 ,66058   ,870,870,870
BEGIN DESCRIPTION:
Verde Creek 117.0
END DESCRIPTION:
XS GIS Cut Line= 3
      1920871.96     13869874.36        1920825.       13869675.
      1920225.03     13869075.03
#Sta/Elev= 30
  4795.5 1708.26  4818.2 1708.37    4846 1710.66  4907.4    1711  4912.4 1710.17
  4916.9  1707.2  4918.6 1704.21    4923 1696.37  4929.9  1690.5  4934.9 1689.61
  4962.3 1688.92  4972.3 1689.85  4984.7 1689.41  4985.7 1687.14  4986.2 1686.64
  4998.9 1687.14  5008.5 1690.32    5021 1690.45  5042.1  1694.2  5105.7 1697.51
  5166.9 1699.54  5173.9 1698.22  5194.8 1697.92  5305.1 1699.09  5445.3 1704.45
  5665.8 1706.45  5698.6 1707.43    5772  1711.1  5810.2 1717.73  5848.8 1728.51
#Mann= 6 ,-1 , 0
  4795.5     .07       0  4918.6      .1       0  4985.7     .05       0
  4998.9      .1       0  5166.9     .07       0  5698.6      .1       0
Bank Sta=4985.7,4998.9
XS Rating Curve= 0 ,0
Exp/Cntr=0.3,0.1

Type RM Length L Ch R = 1 ,65188   ,487,487,487
BEGIN DESCRIPTION:
Verde Creek 116.0
END DESCRIPTION:
XS GIS Cut Line= 5
      1920924.11     13869995.78      1921191.24     13869433.67
      1921157.87     13869101.22      1921133.45     13868990.95
      1920664.93     13868606.95
#Sta/Elev= 30
  3965.4 1706.26  4008.5 1704.36  4210.7 1699.57  4277.5 1699.09  4323.6 1698.86
  4504.4 1698.73  4556.1 1700.33  4643.5 1701.07  4865.6 1697.61  4917.8 1692.86
  4939.1 1692.18  4963.9 1690.49  4994.6 1683.39  5003.8 1682.94  5009.6 1681.22
  5010.1 1680.72  5022.9 1681.22  5081.7 1683.67  5091.5 1685.77  5103.3 1689.92
  5119.6 1690.53    5129 1694.33    5146  1695.4  5151.1 1698.61  5166.9 1700.68
  5362.9  1704.7  5522.1 1708.07  5592.8 1710.84  5618.4 1711.72  5640.6 1712.65
#Mann= 10 ,-1 , 0
  3965.4      .1       0  4008.5     .07       0  4277.5    .035       0
  4323.6     .07       0  4939.1      .1       0  5009.6     .05       0
  5022.9      .1       0  5362.9     .07       0  5592.8      .1       0
  5618.4     .07       0
Bank Sta=5009.6,5022.9
XS Rating Curve= 0 ,0
Exp/Cntr=0.3,0.1

Type RM Length L Ch R = 1 ,64701   ,445,445,445
BEGIN DESCRIPTION:
Verde Creek 115.0
END DESCRIPTION:
XS GIS Cut Line= 4
      1920889.06     13870077.92      1921339.49     13869386.31
        1921525.       13869275.      1921725.04     13869224.99
#Sta/Elev= 30
  3961.9  1710.8  3999.3 1707.31  4098.1 1703.37  4303.4 1698.51  4443.2 1697.22
  4614.5  1698.8    4633 1699.18    4668 1700.16  4741.4 1699.94  4793.1  1695.6
  4810.6 1691.92    4858  1690.8    4877 1683.84    4891 1682.75    4905 1679.76
  4964.5 1680.56  4980.4 1678.57  4980.9 1678.07  4997.5 1678.57  5003.9 1679.31
  5009.6 1680.64  5030.9 1691.57  5049.4  1707.9  5089.6 1733.05  5120.9 1764.49
  5140.6  1781.1  5142.2 1783.17  5145.3 1793.24  5157.1 1803.71  5209.8 1833.33
#Mann= 9 ,-1 , 0
  3961.9      .1       0  4098.1     .07       0  4303.4    .035       0
  4443.2     .07       0  4614.5    .035       0    4633     .07       0
  4980.4     .05       0  4997.5     .07       0  5003.9      .1       0
Bank Sta=4980.4,4997.5
XS Rating Curve= 0 ,0
Exp/Cntr=0.3,0.1

Type RM Length L Ch R = 1 ,64256   ,481,481,481
BEGIN DESCRIPTION:
Verde Creek 114.0
END DESCRIPTION:
XS GIS Cut Line= 3
      1920906.01     13870151.71        1921575.       13869675.
      1921875.01       13869625.
#Sta/Elev= 30
  4182.8 1711.49  4220.2 1709.98    4288 1702.91  4455.5 1697.51    4609 1695.77
  4621.7 1697.01  4652.3 1695.35  4724.8 1695.34  4776.4 1694.45  4820.6 1691.82
  4853.4 1685.49  4905.4 1681.58  4927.5 1677.68  4961.8 1677.51  4988.9 1674.72
  4989.4 1674.22  5006.1 1674.72  5016.9 1678.04  5029.1 1678.34  5035.1 1681.09
  5085.3 1718.37    5099 1734.94  5120.3 1756.15  5135.5 1767.89  5158.3 1778.53
  5260.2 1835.96  5269.3 1841.84  5275.4 1848.95    5286 1856.32  5308.4  1857.6
#Mann= 9 ,-1 , 0
  4182.8      .1       0    4288     .07       0  4455.5    .035       0
    4609     .07       0  4724.8    .035       0  4820.6     .07       0
  4961.8      .1       0  4988.9     .05       0  5006.1      .1       0
Bank Sta=4988.9,5006.1
XS Rating Curve= 0 ,0
Exp/Cntr=0.3,0.1

Type RM Length L Ch R = 1 ,63775   ,329,329,329
BEGIN DESCRIPTION:
Verde Creek 113.0
END DESCRIPTION:
XS GIS Cut Line= 3
      1921153.46     13870268.41        1921575.       13870125.
      1921924.97     13869825.03
#Sta/Elev= 30
  4559.3 1698.29  4767.4 1692.85  4780.1 1690.67  4799.1 1690.51    4844 1684.23
  4935.3 1676.61  4953.1 1673.96    4967 1675.14  4973.4 1674.13    4986    1675
  4986.9 1673.85  4987.4 1673.35  5004.1 1673.85  5004.6 1674.82  5013.4 1675.23
  5068.9 1675.88    5078 1676.15  5084.2 1677.82  5092.1 1684.38    5096 1688.99
    5100 1691.26  5151.4 1703.87  5202.7 1723.91  5222.5 1735.15  5277.8 1762.13
  5336.1 1784.39  5368.7 1801.75  5416.1 1831.15  5437.5 1842.56  5465.5 1854.83
#Mann= 5 ,-1 , 0
  4559.3    .035       0  4953.1     .07       0  4986.9     .05       0
  5004.1     .07       0  5068.9      .1       0
Bank Sta=4986.9,5004.1
XS Rating Curve= 0 ,0
Exp/Cntr=0.3,0.1

Type RM Length L Ch R = 1 ,63446   ,580,580,580
BEGIN DESCRIPTION:
Verde Creek 112.0
END DESCRIPTION:
XS GIS Cut Line= 3
      1921274.32     13870555.03      1921706.66     13870411.54
      1922025.03     13869924.96
#Sta/Elev= 30
  4585.9 1700.64  4606.4 1699.61  4631.4 1695.69  4665.7 1696.08  4719.9 1691.38
  4759.8 1690.06  4824.2 1680.05  4846.3 1679.07  4871.6 1674.95  4945.1 1672.63
  4970.4 1670.73  4970.9 1670.23  4987.6 1670.73  5004.3 1674.82  5029.6 1687.13
  5046.6 1689.78  5070.3 1691.51    5158 1692.24  5246.2 1696.76  5261.7 1698.85
  5268.8 1701.87  5283.2 1702.88  5292.2 1707.93  5307.6 1712.32  5340.5 1722.56
  5354.9 1728.76  5365.6 1729.92  5487.5 1779.59  5566.4 1809.77  5622.9  1829.6
#Mann= 6 ,-1 , 0
  4585.9    .035       0  4945.1      .1       0  4970.4     .05       0
  4987.6      .1       0  5246.2    .035       0  5307.6      .1       0
Bank Sta=4970.4,4987.6
XS Rating Curve= 0 ,0
Exp/Cntr=0.3,0.1

Type RM Length L Ch R = 1 ,62866   ,477,477,477
BEGIN DESCRIPTION:
Verde Creek 111.0
END DESCRIPTION:
XS GIS Cut Line= 4
      1921674.97     13871075.03        1921825.       13870925.
      1921955.52     13870746.47      1922053.94     13870118.57
#Sta/Elev= 30
  4788.1 1707.04  4849.5  1703.4  4906.2 1698.62  4922.2 1692.71  4931.7 1682.52
  4937.5 1674.93  4943.4 1671.79  4959.2 1670.56  4978.3 1670.12  4986.6 1667.91
  4987.1 1667.41  5003.9 1667.91  5017.3 1669.83  5050.2 1670.42  5080.5 1680.49
  5102.8 1683.69  5136.2 1685.72  5209.2 1686.68  5340.1 1690.02  5445.9 1689.19
  5548.3 1690.53  5701.4 1696.68  5725.7 1698.64  5753.5    1704  5768.3 1709.18
  5774.3 1713.48  5779.8 1713.91  5789.5 1714.15  5803.9 1722.88    5857 1743.37
#Mann= 9 ,-1 , 0
  4788.1     .07       0  4849.5    .035       0  4931.7     .07       0
  4959.2      .1       0  4986.6     .05       0  5003.9      .1       0
  5209.2     .07       0  5445.9    .035       0  5779.8      .1       0
Bank Sta=4986.6,5003.9
XS Rating Curve= 0 ,0
Exp/Cntr=0.3,0.1

Type RM Length L Ch R = 1 ,62389   ,445,445,445
BEGIN DESCRIPTION:
Verde Creek 110.0
END DESCRIPTION:
XS GIS Cut Line= 3
        1922225.     13871225.03        1922225.       13871025.
      1922136.29     13870118.96
#Sta/Elev= 30
  4800.4    1717  4802.8 1717.01  4866.7 1712.35  4880.2 1709.53  4887.7 1703.65
  4892.2 1694.65  4904.2 1682.27  4916.2 1674.37  4934.8 1668.25  4950.6 1665.31
  4979.2 1667.36  5000.5 1664.56    5001 1664.06    5018 1664.56  5018.3 1666.05
  5019.7 1666.04  5064.8 1667.17  5075.5 1672.02    5084 1673.58  5232.4 1678.76
  5289.6 1686.01  5358.6 1686.89  5556.2 1687.38  5777.7  1694.9    5811 1696.49
  5849.3 1703.05  5877.4 1712.27  5892.4 1721.13  5904.5 1721.84  5910.8  1726.2
#Mann= 9 ,-1 , 0
  4800.4     .07       0  4802.8     .07       0  4934.8      .1       0
  5000.5     .05       0    5018      .1       0  5019.7     .07       0
  5358.6     .07       0  5777.7     .07       0  5849.3      .1       0
Bank Sta=5000.5,5018
XS Rating Curve= 0 ,0
Exp/Cntr=0.3,0.1

Type RM Length L Ch R = 1 ,61944   ,419,419,419
BEGIN DESCRIPTION:
Verde Creek 109.0
END DESCRIPTION:
XS GIS Cut Line= 4
      1922575.01     13870925.02        1922525.       13870725.
        1922475.       13870525.      1922245.24     13869998.15
#Sta/Elev= 30
  4798.2 1693.79    4810 1692.29  4855.7 1690.35  4874.3 1687.98    4899 1683.19
  4911.4 1677.25  4926.3 1675.96  4951.6  1665.6  4981.8 1661.79  4982.3 1661.29
  4999.4 1661.79  5010.3 1662.51  5025.2 1665.59  5078.3 1666.68  5112.4 1675.43
  5120.9 1676.24  5129.1 1676.66  5146.4 1683.16  5164.9 1684.36  5427.4 1685.41
  5558.3 1689.63  5634.7 1693.44  5649.9 1696.99  5664.3 1698.48  5686.7 1706.83
  5728.1 1723.79  5741.6 1730.43  5754.7 1734.93  5771.4 1744.05  5785.3 1745.77
#Mann= 6 ,-1 , 0
  4798.2      .1       0  4981.8     .05       0  4999.4      .1       0
  5120.9     .07       0  5427.4     .07       0  5686.7      .1       0
Bank Sta=4981.8,4999.4
XS Rating Curve= 0 ,0
Exp/Cntr=0.3,0.1

Type RM Length L Ch R = 1 ,61525   ,490,490,490
BEGIN DESCRIPTION:
Verde Creek 108.0
END DESCRIPTION:
XS GIS Cut Line= 3
        1922875.     13871025.01        1922825.       13870475.
        1922225.       13869875.
#Sta/Elev= 30
  4442.9 1708.55  4459.6 1706.71  4572.2  1694.1  4620.8 1684.85  4756.8 1674.46
  4804.9 1670.94  4825.2 1671.46  4879.5 1665.61  4966.8 1663.04  4999.6 1664.18
  5031.3 1660.84  5031.8 1660.34  5048.9 1660.84  5065.4 1665.74  5078.1 1672.59
  5101.5 1674.71    5129 1681.89    5203 1683.07  5358.1 1683.75  5502.5 1687.99
  5570.3 1691.49  5602.1 1694.89  5626.9 1700.93  5667.7 1715.56  5697.5  1729.3
  5742.1 1744.92  5773.8 1760.23  5790.7 1762.46  5799.4 1768.88  5843.7 1789.13
#Mann= 8 ,-1 , 0
  4442.9    .035       0  4459.6     .07       0  4620.8    .035       0
  4756.8      .1       0  5031.3     .05       0  5048.9      .1       0
    5203     .07       0  5626.9      .1       0
Bank Sta=5031.3,5048.9
XS Rating Curve= 0 ,0
Exp/Cntr=0.3,0.1
