HEC-RAS study Verde Creek.prj: Verde Creek Base Level Engineering

--- Verde Creek.g01 (geometry) --- (continued)

Type RM Length L Ch R = 1 ,61035   ,448,448,448
BEGIN DESCRIPTION:
Verde Creek 107.0
END DESCRIPTION:
XS GIS Cut Line= 3
      1923337.09     13870943.91        1923275.       13870375.
       1922727.1     13869103.19
#Sta/Elev= 30
  4427.8  1704.7  4590.4 1687.87  4780.6 1678.56  4807.7 1675.95  4827.7 1670.91
  4844.4 1666.84  4873.8 1664.55  4931.4 1662.85  4967.7 1660.33  4980.4 1656.15
  5001.9 1655.94  5002.4 1655.44  5019.5 1655.94  5020.5 1659.81  5022.4 1660.31
  5046.6 1662.65  5061.2 1672.16  5074.1 1677.48  5092.4 1679.52  5392.9 1678.81
  5645.7 1683.77  5918.8 1694.02  5988.9 1700.26  6026.9 1703.22  6118.1 1716.07
  6186.9 1734.15  6238.9 1750.86  6287.9 1761.53  6368.8 1787.62  6384.9 1790.92
#Mann= 8 ,-1 , 0
  4427.8    .035       0  4827.7      .1       0  4844.4     .07       0
  4873.8      .1       0  5001.9     .05       0  5019.5      .1       0
  5074.1     .07       0  5988.9      .1       0
Bank Sta=5001.9,5019.5
XS Rating Curve= 0 ,0
Exp/Cntr=0.3,0.1

Type RM Length L Ch R = 1 ,60587   ,487,487,487
BEGIN DESCRIPTION:
Verde Creek 106.0
END DESCRIPTION:
XS GIS Cut Line= 5
      1923518.44     13871234.96      1923664.47     13870750.39
        1923675.       13870225.      1923565.25     13869488.84
      1923473.07     13868994.14
#Sta/Elev= 30
    3968 1723.42  4149.4 1710.05  4194.2 1703.81    4328 1690.69  4571.2 1678.48
  4742.5 1677.65  4850.3 1677.11  4877.4 1671.43  4896.2 1657.77  4910.3 1655.55
  4988.6 1653.68  4989.1 1653.18  5006.2 1653.68  5007.8 1658.41  5018.6 1662.86
  5077.4  1673.9  5100.5 1676.93  5418.1 1675.72  5696.8 1677.91  5734.4 1678.22
  5762.2 1682.87  5789.3 1676.34  5810.6 1673.91  5959.3 1683.43  5987.6 1695.63
  6018.1 1712.11  6140.2 1761.23  6171.2 1776.05  6182.9 1778.77  6247.1 1809.75
#Mann= 11 ,-1 , 0
    3968    .035       0  4194.2     .07       0  4571.2    .035       0
  4742.5     .07       0  4896.2      .1       0  4988.6     .05       0
  5006.2      .1       0  5077.4     .07       0  5696.8      .1       0
  5810.6     .07       0  5959.3      .1       0
Bank Sta=4988.6,5006.2
XS Rating Curve= 0 ,0
Exp/Cntr=0.3,0.1

Type RM Length L Ch R = 1 ,60100   ,450,450,450
BEGIN DESCRIPTION:
Verde Creek 105.0
END DESCRIPTION:
XS GIS Cut Line= 4
      1923966.14     13870968.48      1924155.47     13870484.74
        1924125.       13870125.      1923794.75     13869533.33
#Sta/Elev= 30
  4119.1 1683.53  4218.1 1679.92  4456.3 1672.53  4646.4 1672.44  4901.8 1674.32
  4939.4 1670.41  4951.2    1668  4957.2 1662.63  4960.2 1657.72  4963.2 1655.14
  4975.3 1651.34  4981.3 1651.29  4981.8 1650.13  4982.3 1649.63  4999.5 1650.13
    5030 1650.77    5041 1653.16  5078.3 1653.94  5097.2 1659.41  5115.9 1663.58
  5135.8 1662.55  5155.6 1668.21  5171.1 1670.48  5188.3 1670.73  5198.6 1669.14
    5224 1672.71  5250.1 1674.51  5346.3 1672.92    5418 1673.04  5677.2 1679.81
#Mann= 7 ,-1 , 0
  4119.1     .07       0  4218.1    .035       0  4456.3     .07       0
  4939.4      .1       0  4981.8     .05       0  4999.5      .1       0
  5097.2     .07       0
Bank Sta=4981.8,4999.5
XS Rating Curve= 0 ,0
Exp/Cntr=0.3,0.1

Type RM Length L Ch R = 1 ,59650   ,455,455,455
BEGIN DESCRIPTION:
Verde Creek 104.0
END DESCRIPTION:
XS GIS Cut Line= 4
       1924252.4     13870926.52      1924527.27      13870247.6
        1924525.       13869975.      1924507.21     13869185.76
#Sta/Elev= 30
  3994.9 1678.59  4233.2 1671.82  4312.2 1669.58  4831.7 1673.02  4878.3  1668.2
  4915.7 1663.78  4921.7 1662.28  4936.7 1653.57  4957.7 1649.39  5032.7 1648.42
  5033.2 1647.92  5050.7 1648.42  5053.1 1651.34  5074.7  1660.7  5101.7 1667.59
  5149.8 1669.14  5293.9 1677.96  5407.5 1691.21  5422.8 1691.57  5434.8 1694.15
  5527.9  1725.8  5575.9 1745.45  5632.9 1772.36  5677.9  1798.1  5725.9 1830.33
  5728.9 1833.77  5731.9 1841.52  5737.9 1847.29  5752.9 1850.17  5789.4 1851.94
#Mann= 5 ,-1 , 0
  3994.9    .035       0  4233.2     .07       0  4878.3      .1       0
  5032.7     .05       0  5050.7      .1       0
Bank Sta=5032.7,5050.7
XS Rating Curve= 0 ,0
Exp/Cntr=0.3,0.1

Type RM Length L Ch R = 1 ,59195   ,443,443,443
BEGIN DESCRIPTION:
Verde Creek 103.0
END DESCRIPTION:
XS GIS Cut Line= 3
      1924775.03     13870174.97        1924925.       13870025.
      1925275.01       13869925.
#Sta/Elev= 30
  4792.5 1670.17    4852 1669.98    4918  1662.8  4943.4  1657.1  4981.4 1645.27
  4993.9 1645.04  5000.2 1643.46  5000.7 1642.96  5018.2 1643.46  5031.1 1647.45
  5061.5 1647.56  5090.3 1652.78  5130.9 1663.34  5143.4 1670.93  5155.9 1674.82
  5168.3 1681.59  5177.7 1684.85  5207.6 1701.47  5227.6 1717.98    5245 1729.68
  5252.6 1739.49  5255.7 1741.76  5274.4 1761.84  5288.7 1772.56  5305.8 1790.99
  5308.1 1794.57    5315 1848.03  5316.8 1851.66  5331.8 1853.75  5368.6 1853.72
#Mann= 4 ,-1 , 0
  4792.5    .035       0  5000.2    .035       0  5018.2    .035       0
  5061.5      .1       0
Bank Sta=5000.2,5018.2
XS Rating Curve= 0 ,0
Exp/Cntr=0.3,0.1

Type RM Length L Ch R = 1 ,58752   ,475,475,475
BEGIN DESCRIPTION:
Verde Creek 102.0
END DESCRIPTION:
XS GIS Cut Line= 3
      1924674.98       13870425.        1924875.       13870425.
        1925325.       13870075.
#Sta/Elev= 30
  4796.3 1668.63  4966.8 1668.85  4981.8 1666.28  4984.8 1664.67  4989.2 1659.45
  4996.3 1650.55  5004.5 1643.75  5017.4 1641.28  5017.9 1640.78  5035.4 1641.28
  5091.9 1645.03  5232.5 1648.36  5245.1 1649.64  5254.9 1653.39  5264.7 1653.01
  5270.5 1655.02  5289.5 1656.52  5297.1 1658.55  5372.2 1696.22  5388.4 1707.32
  5416.2 1721.73  5440.6 1737.41  5468.2 1758.57  5474.8 1764.91  5494.6 1778.29
  5521.4 1802.56  5525.2  1809.9    5529 1839.15  5532.8 1850.82  5566.4  1852.8
#Mann= 4 ,-1 , 0
  4796.3     .07       0  4989.2      .1       0  5017.4     .05       0
  5035.4      .1       0
Bank Sta=5017.4,5035.4
XS Rating Curve= 0 ,0
Exp/Cntr=0.3,0.1

Type RM Length L Ch R = 1 ,58277   ,660,660,660
BEGIN DESCRIPTION:
Verde Creek 101.0
END DESCRIPTION:
XS GIS Cut Line= 4
      1924499.45     13870771.94       1925054.1     13870791.98
      1925307.39     13870719.73      1925474.99     13870175.03
#Sta/Elev= 30
    4293 1670.85  4453.2 1669.06  4551.7 1667.96  4666.2 1666.56  4693.3 1662.11
  4729.8 1661.55  4748.7 1657.53  4765.3 1651.74  4807.3 1661.93  4847.2    1664
  4874.4 1663.11  4895.7 1649.43  4911.8 1643.34  4983.6 1641.36  5005.7 1636.78
  5006.2 1636.28  5023.8 1636.78    5074 1646.19  5121.3 1646.86  5139.9 1649.35
  5237.5 1655.44  5267.9 1659.32    5294  1665.2  5320.8 1676.12    5341 1685.99
  5425.8  1734.7  5488.6 1762.19  5598.4 1816.25  5645.5 1836.81  5681.3 1845.91
#Mann= 9 ,-1 , 0
    4293    .035       0  4453.2     .07       0  4551.7    .035       0
  4748.7     .07       0  4847.2      .1       0  5005.7     .05       0
  5023.8      .1       0  5139.9    .035       0  5320.8      .1       0
Bank Sta=5005.7,5023.8
XS Rating Curve= 0 ,0
Exp/Cntr=0.3,0.1

Type RM Length L Ch R = 1 ,57617   ,535,535,535
BEGIN DESCRIPTION:
Verde Creek 100.0
END DESCRIPTION:
XS GIS Cut Line= 4
      1925325.09     13871824.82        1925575.       13871325.
        1925775.       13870925.        1925725.     13870275.05
#Sta/Elev= 30
  3998.1 1663.82  4052.9  1663.6  4408.1 1663.85    4486 1661.32  4594.3 1657.15
  4633.8  1648.8  4682.4 1648.01  4702.6 1647.16  4810.8  1643.3  4909.1 1638.42
  4952.4 1637.97  4958.2 1636.96  4963.9 1631.82  4964.4 1631.32  4994.6 1631.82
    4996 1634.56  5025.4 1637.27    5051 1641.91  5105.2 1662.03  5204.5 1662.62
  5279.1 1665.76  5301.5 1675.28  5322.1 1677.47  5337.1  1684.4  5342.9 1688.14
  5345.9 1694.52  5351.8  1698.5  5487.3 1767.26  5601.6 1819.32    5656  1836.4
#Mann= 14 ,-1 , 0
  3998.1      .1       0  4052.9    .035       0    4486      .1       0
  4594.3     .07       0  4682.4    .035       0  4702.6     .07       0
  4810.8      .1       0  4909.1     .07       0  4963.9     .05       0
  4994.6     .07       0  5025.4      .1       0  5204.5    .035       0
  5322.1     .07       0  5337.1      .1       0
Bank Sta=4963.9,4994.6
XS Rating Curve= 0 ,0
Exp/Cntr=0.3,0.1

Type RM Length L Ch R = 1 ,57082   ,518,518,518
BEGIN DESCRIPTION:
Verde Creek 99.0
END DESCRIPTION:
XS GIS Cut Line= 4
      1926022.28     13871985.87        1926125.       13871575.
        1926225.       13871175.      1926253.92     13870108.82
#Sta/Elev= 30
  4159.2 1662.47  4352.2 1660.57  4450.5 1658.97  4481.5 1653.65  4487.6 1657.57
  4592.8 1660.25  4617.5 1657.32  4660.8  1648.8    4667 1645.65  4787.6 1640.32
  4855.2 1639.83    4936 1640.21    4967 1637.22  4992.7  1631.7  5009.4 1631.58
  5009.9 1631.08  5040.2 1631.58  5051.8 1635.82  5085.8 1633.07  5105.8 1639.85
  5132.8 1643.49  5171.9 1654.43  5192.8 1657.41  5614.3 1659.92  5783.7  1668.6
  5910.1 1674.91  5932.1 1679.75  5986.6 1699.36  6009.8  1707.9  6061.6 1727.71
#Mann= 9 ,-1 , 0
  4159.2    .035       0  4352.2     .07       0  4855.2      .1       0
  5009.4     .05       0  5040.2      .1       0  5192.8    .035       0
  5783.7     .07       0  5986.6      .1       0  6009.8     .07       0
Bank Sta=5009.4,5040.2
XS Rating Curve= 0 ,0
Exp/Cntr=0.3,0.1

Type RM Length L Ch R = 1 ,56564   ,488,488,488
BEGIN DESCRIPTION:
Verde Creek 98.0
END DESCRIPTION:
XS GIS Cut Line= 5
        1926675.      13872136.6        1926675.       13871775.
        1926675.       13871375.        1926675.       13870975.
      1926521.07     13870071.82
#Sta/Elev= 30
  4233.1 1665.11  4238.1 1665.09  4337.3 1663.77  4748.6 1657.89  4846.9 1655.66
  4864.5 1652.62  4891.5 1638.89  4909.5 1632.75  4932.8 1632.85  4954.5 1631.48
  4987.5 1633.42  4993.5 1632.94    4996 1630.21  4996.5 1629.71    5027 1630.21
    5062 1637.46  5080.5 1636.51  5104.9 1638.72  5149.5 1647.55    5197 1650.13
  5272.5 1654.75  5394.7 1657.41  6091.7 1658.08  6147.2 1660.75  6171.5 1666.14
  6198.4 1676.96  6240.8 1703.21  6255.6 1713.09    6278 1722.45  6310.9  1730.5
#Mann= 11 ,-1 , 0
  4233.1     .07       0  4238.1    .035       0  4337.3      .1       0
  4748.6    .035       0  4846.9     .07       0  4932.8      .1       0
    4996     .05       0    5027      .1       0    5197    .035       0
  6091.7     .07       0  6240.8      .1       0
Bank Sta=4996,5027
XS Rating Curve= 0 ,0
Exp/Cntr=0.3,0.1

Type RM Length L Ch R = 1 ,56076   ,537,537,537
BEGIN DESCRIPTION:
Verde Creek 97.0
END DESCRIPTION:
XS GIS Cut Line= 3
        1927025.     13871724.98        1927075.       13871325.
      1926969.73     13870497.06
#Sta/Elev= 30
  4592.4 1660.31  4685.5 1659.28  4784.2 1657.67    4883  1656.5  4898.5 1655.21
  4902.5 1652.05  4904.5 1647.44  4907.6 1644.11  4922.2 1640.12  4933.6 1633.26
  4940.8 1630.93  4950.9 1629.26  4995.3 1629.99  4998.3 1628.68  5009.2 1628.36
    5010 1627.51  5010.5 1627.01    5041 1627.51  5043.6 1630.92  5061.8 1632.22
  5073.9 1634.88  5106.5 1637.17  5122.3 1639.19  5151.4  1640.2  5231.9 1646.28
  5280.2  1650.9  5349.1 1654.59    5425 1656.04  5672.7 1654.76  5830.1 1656.03
#Mann= 7 ,-1 , 0
  4592.4     .07       0  4685.5      .1       0  4784.2    .035       0
    4883      .1       0    5010     .05       0    5041      .1       0
  5106.5    .035       0
Bank Sta=5010,5041
XS Rating Curve= 0 ,0
Exp/Cntr=0.3,0.1

Type RM Length L Ch R = 1 ,55539   ,239,239,239
BEGIN DESCRIPTION:
Verde Creek 96.0
END DESCRIPTION:
XS GIS Cut Line= 3
      1927563.61     13871713.44        1927525.       13871075.
      1927077.23     13870490.63
#Sta/Elev= 30
  4360.4 1658.42  4714.1 1653.65  4764.3 1652.05  4772.6 1651.13  4788.3 1651.27
  4824.4 1648.44  4848.5 1645.39  4890.6 1637.49  4905.6 1633.34  4911.6 1630.92
  4920.6 1629.13  4930.1 1629.17  4939.8 1629.28  4951.2 1628.13  4959.7 1628.87
  4968.2 1627.29  4968.7 1626.79  4999.3 1627.29  5001.6 1628.46  5035.4 1629.72
  5059.4 1632.63    5083  1634.4  5130.7 1643.44  5149.2 1648.44    5161 1651.32
  5198.5 1652.49  5213.5 1651.98  5319.2 1653.69  5356.9 1654.52  5736.2 1655.61
#Mann= 8 ,-1 , 0
  4360.4     .07       0  4714.1    .035       0  4788.3     .07       0
  4930.1      .1       0  4968.2     .05       0  4999.3      .1       0
  5149.2     .07       0  5319.2    .035       0
Bank Sta=4968.2,4999.3
XS Rating Curve= 0 ,0
Exp/Cntr=0.3,0.1

Type RM Length L Ch R = 1 ,55300   ,311,311,311
BEGIN DESCRIPTION:
Verde Creek 95.1
END DESCRIPTION:
XS GIS Cut Line= 3
      1928172.01     13872087.44      1927999.13     13871278.73
      1927367.87     13870616.88
#Sta/Elev= 30
  3799.5 1662.35  4005.6 1659.61  4023.6 1660.35  4173.4  1654.3  4331.9 1650.99
  4433.2 1647.34  4467.6  1645.1    4516 1645.57  4621.9 1637.53  4676.8 1635.93
  4691.7 1634.56  4703.2 1630.82  4708.6 1632.25  4721.4 1641.23    4728 1644.01
  4742.6    1647  4771.5 1648.32  4833.8 1645.28  4913.1 1636.67  4918.1 1636.11
  4979.5  1629.4  5029.2 1627.58  5029.7 1627.08  5060.3 1627.58  5065.1 1629.84
  5127.3 1636.41  5184.1 1651.79  5229.7 1653.52  5434.1  1653.5  5541.1  1654.7
#Mann= 11 ,-1 , 0
  3799.5     .07       0  4005.6    .035       0  4331.9     .07       0
  4433.2    .035       0    4516     .07       0  4771.5    .035       0
  4913.1     .07       0  4918.1      .1       0  5029.2     .05       0
  5060.3      .1       0  5434.1    .035       0
Bank Sta=5029.2,5060.3
XS Rating Curve= 0 ,0
Exp/Cntr=0.3,0.1

Type RM Length L Ch R = 1 ,54989   ,541,541,541
BEGIN DESCRIPTION:
Verde Creek 95.0
END DESCRIPTION:
XS GIS Cut Line= 4
      1928251.57     13872218.16      1928154.21     13871269.55
        1928025.       13870925.       1928094.4     13870347.43
#Sta/Elev= 30
  3679.1 1664.13  3954.4  1660.3  4000.7 1661.12  4032.2 1656.37  4329.9 1655.43
  4353.2  1653.5  4429.1 1653.33  4610.9 1650.21  4685.4 1643.67    4743 1633.92
  4775.7 1632.63  4789.6 1628.82  4793.2 1630.08  4822.3 1636.46  4839.9 1637.94
    4900 1635.62  4946.2 1630.99  4973.7 1627.67  5002.7 1627.72  5017.6 1624.78
  5030.8 1624.41  5031.4 1623.91  5064.8 1624.41  5065.9 1626.63  5087.1 1627.92
  5182.4 1645.78    5212 1648.86  5429.4 1652.65  5554.4 1654.26  5582.4 1654.64
#Mann= 15 ,-1 , 0
  3679.1     .07       0  3954.4      .1       0  4032.2    .035       0
  4329.9     .07       0  4353.2    .035       0  4429.1     .07       0
  4793.2    .035       0  4839.9     .07       0  4946.2      .1       0
  5030.8     .05       0  5064.8      .1       0  5182.4    .035       0
    5212      .1       0  5429.4     .07       0  5554.4      .1       0
Bank Sta=5030.8,5064.8
XS Rating Curve= 0 ,0
Exp/Cntr=0.3,0.1

Type RM Length L Ch R = 1 ,54448   ,605,605,605
BEGIN DESCRIPTION:
Verde Creek 94.0
END DESCRIPTION:
XS GIS Cut Line= 4
      1928992.83     13872047.81      1928831.87     13871282.06
        1928425.       13870725.      1928225.01     13870375.02
#Sta/Elev= 30
  3527.2 1658.94  3581.9 1659.25    3857 1655.09  3991.6 1652.78  4309.7 1648.35
  4374.8 1648.06  4395.2 1648.94  4432.9 1647.74    4550 1646.66  4615.4 1646.06
  4653.7 1644.71    4666 1643.28  4698.3 1636.69  4713.2 1632.59    4728 1632.74
  4790.7 1629.82  4864.5 1626.62  4895.2 1626.47  4924.1 1624.46  4969.7 1625.03
  4976.9 1624.73  4984.6 1622.82  4985.4 1622.32  5020.8 1622.82  5021.7 1627.89
  5043.7 1634.78  5092.5 1646.65  5113.9 1648.81  5254.8 1652.08  5402.6 1653.62
#Mann= 10 ,-1 , 0
  3527.2     .05       0    3857     .07       0  3991.6    .035       0
    4550      .1       0    4666    .035       0  4790.7      .1       0
  4984.6     .05       0  5020.8      .1       0  5113.9    .035       0
  5254.8     .07       0
Bank Sta=4984.6,5020.8
XS Rating Curve= 0 ,0
Exp/Cntr=0.3,0.1

Type RM Length L Ch R = 1 ,53843   ,471,471,471
BEGIN DESCRIPTION:
Verde Creek 93.0
END DESCRIPTION:
XS GIS Cut Line= 5
      1929029.56     13872067.87      1928901.85     13870962.48
      1928968.02     13870724.43      1929077.36     13870521.27
      1929675.03     13870024.97
#Sta/Elev= 30
  3640.9 1658.68    3899 1656.03  4010.7 1654.31  4354.4 1650.09  4425.6 1648.94
  4515.9 1647.48  4706.2 1645.89  4914.2 1625.83  4965.6 1623.05  4969.2 1619.94
  4970.1 1619.44  5005.5 1619.94  5020.4 1622.23  5078.1 1624.59  5098.6 1632.66
  5115.6 1644.96  5197.4 1636.23    5238 1639.15  5396.4 1651.42  5534.7 1658.45
  5602.2 1661.69  5659.6 1669.04  5766.8 1692.93  5791.2 1701.23  5836.6 1714.54
  5863.5 1727.45  5884.7 1731.28  5939.6 1742.57  5976.6 1749.21  6008.3 1751.27
#Mann= 17 ,-1 , 0
  3640.9     .05       0    3899     .07       0  4010.7     .05       0
  4354.4    .035       0  4425.6     .05       0  4515.9    .035       0
  4914.2      .1       0  4969.2     .05       0  5005.5      .1       0
  5020.4     .07       0    5238    .035       0  5396.4     .07       0
  5534.7      .1       0  5659.6    .035       0  5791.2      .1       0
  5884.7    .035       0  5939.6      .1       0
Bank Sta=4969.2,5005.5
XS Rating Curve= 0 ,0
Exp/Cntr=0.3,0.1

Type RM Length L Ch R = 1 ,53372   ,585,585,585
BEGIN DESCRIPTION:
Verde Creek 92.0
END DESCRIPTION:
XS GIS Cut Line= 4
       1929102.2     13872104.67        1929279.     13870942.65
        1929425.       13870775.      1929924.98     13870175.02
#Sta/Elev= 30
  3606.7 1658.26  3836.7 1656.22  4437.5 1645.19    4610 1643.72  4686.4 1644.56
    4709 1640.66    4744 1639.71  4774.4 1635.49  4883.4 1627.55  4942.4  1619.1
  4955.2 1619.02    4956 1618.52  4991.6 1619.02  4995.4  1621.1  5027.4 1622.38
  5076.9 1634.47  5099.1 1638.03  5148.8 1642.21    5193 1643.63  5267.6 1647.17
  5293.6 1649.55  5303.4 1654.54  5379.4 1676.83  5436.2 1698.93  5511.5 1731.47
  5584.6 1769.88  5705.7 1827.38  5717.4 1835.18  5736.4 1844.54  5785.4 1847.57
#Mann= 9 ,-1 , 0
  3606.7     .05       0    4610    .035       0    4709     .07       0
  4942.4      .1       0  4955.2     .05       0  4991.6      .1       0
    5193     .07       0  5267.6    .035       0  5379.4      .1       0
Bank Sta=4955.2,4991.6
XS Rating Curve= 0 ,0
Exp/Cntr=0.3,0.1

Type RM Length L Ch R = 1 ,52787   ,534,534,534
BEGIN DESCRIPTION:
Verde Creek 91.0
END DESCRIPTION:
XS GIS Cut Line= 4
      1930231.59      13871933.3      1929943.74     13871218.82
        1929975.       13870875.        1929975.     13870225.03
#Sta/Elev= 30
  3883.8 1656.01  4020.7 1653.77  4214.3 1651.61  4248.2 1648.56  4264.4  1649.7
  4545.1 1641.39  4653.1 1637.86  4738.3 1634.77    4752    1635  4764.1 1630.31
  4836.8 1626.84  4929.8 1622.31  4947.5 1618.57  4948.4 1618.07  4984.4 1618.57
    5038 1621.44    5050 1627.05    5056 1632.04    5071 1637.56    5089 1640.27
  5132.2  1641.7    5203 1645.08  5230.5 1654.38  5266.4 1666.45    5320 1688.43
    5383 1711.35    5425 1729.69    5509 1770.36    5602 1820.83  5649.3 1843.17
#Mann= 10 ,-1 , 0
  3883.8     .07       0  4020.7    .035       0  4545.1     .07       0
  4653.1    .035       0  4738.3     .07       0  4836.8      .1       0
  4947.5     .05       0  4984.4      .1       0  5132.2    .035       0
  5230.5      .1       0
Bank Sta=4947.5,4984.4
XS Rating Curve= 0 ,0
Exp/Cntr=0.3,0.1

Type RM Length L Ch R = 1 ,52253   ,564,564,564
BEGIN DESCRIPTION:
Verde Creek 90.0
END DESCRIPTION:
XS GIS Cut Line= 3
      1930294.15     13871907.65        1930425.       13870975.
        1930525.     13870175.01
#Sta/Elev= 30
  4062.6 1655.34  4359.1 1648.45  4420.4 1648.54  4564.2  1640.8  4674.9 1636.79
  4699.1 1633.25  4729.6 1632.23  4828.5 1625.97  4862.7 1622.77    4887 1616.76
  4920.3 1619.31  4973.1 1615.98    4974 1615.48    5010 1615.98  5011.2 1617.73
  5032.3 1619.94  5059.5 1633.44  5067.8 1635.13  5105.9 1639.11  5223.8 1640.11
  5289.3 1642.21  5308.4 1646.54  5322.5 1647.24  5329.9 1649.38  5385.7  1675.4
  5525.1 1731.73  5673.3 1800.69  5742.8 1835.64  5788.2 1851.55  5810.6 1854.07
#Mann= 8 ,-1 , 0
  4062.6     .07       0  4564.2    .035       0  4729.6     .07       0
  4828.5      .1       0  4973.1     .05       0    5010      .1       0
  5223.8    .035       0  5322.5      .1       0
Bank Sta=4973.1,5010
XS Rating Curve= 0 ,0
Exp/Cntr=0.3,0.1

Type RM Length L Ch R = 1 ,51689   ,553,553,553
BEGIN DESCRIPTION:
Verde Creek 89.0
END DESCRIPTION:
XS GIS Cut Line= 3
      1930839.31     13872097.51        1930925.       13871175.
        1930725.     13870375.01
#Sta/Elev= 30
  4077.7 1655.92  4435.2 1648.93  4681.5  1638.1  4725.8 1633.24    4784 1629.56
    4796 1625.69  4816.3  1625.5  4859.3 1619.88  4914.8 1616.93  4943.8  1613.6
  4973.8 1614.74  4978.1 1612.48    4979 1611.98    5015 1612.48  5015.8 1614.77
  5050.3 1622.09  5071.9  1630.7  5087.4 1634.15  5124.5 1637.82  5218.1    1639
  5258.6 1638.83  5320.3 1638.62  5422.6 1638.91  5489.4  1640.2  5524.8 1646.18
  5535.8 1649.06  5594.5 1679.47  5678.8 1712.16  5773.9 1754.58  5828.8 1776.06
#Mann= 11 ,-1 , 0
  4077.7     .07       0  4725.8    .035       0  4816.3     .07       0
  4914.8      .1       0  4978.1     .05       0    5015      .1       0
  5218.1     .07       0  5258.6      .1       0  5320.3     .07       0
  5422.6    .035       0  5524.8      .1       0
Bank Sta=4978.1,5015
XS Rating Curve= 0 ,0
Exp/Cntr=0.3,0.1

Type RM Length L Ch R = 1 ,51136   ,553,553,553
BEGIN DESCRIPTION:
Verde Creek 88.0
END DESCRIPTION:
XS GIS Cut Line= 4
        1931425.     13871724.98        1931425.       13871325.
        1931125.       13870525.      1931030.47     13870272.92
#Sta/Elev= 30
    4600 1643.94  4760.3 1642.26  4783.7 1640.16  4810.7 1630.36  4822.7 1628.28
  4854.2 1628.14  4897.7 1616.86  4981.7 1614.13  5005.6 1608.31  5006.5 1607.81
  5042.7 1608.31  5044.5 1613.18  5070.2 1616.99  5089.4 1628.07    5099 1630.78
  5134.2 1629.82  5159.9 1633.27  5233.6 1636.64  5385.4 1637.69  5580.2 1639.05
  5686.5 1646.86  5701.4 1646.82  5765.4 1657.29  5836.4  1680.6    5863 1688.93
  5930.6 1702.48  6005.7 1725.53  6036.4 1731.69    6073 1741.68  6123.6  1752.1
#Mann= 10 ,-1 , 0
    4600     .07       0  4760.3    .035       0  4854.2      .1       0
  5005.6     .05       0  5042.7      .1       0  5385.4     .07       0
  5580.2    .035       0  5686.5      .1       0  5836.4    .035       0
  6036.4      .1       0
Bank Sta=5005.6,5042.7
XS Rating Curve= 0 ,0
Exp/Cntr=0.3,0.1

Type RM Length L Ch R = 1 ,50583   ,561,561,561
BEGIN DESCRIPTION:
Verde Creek 87.0
END DESCRIPTION:
XS GIS Cut Line= 4
        1931925.     13871875.02        1931925.       13871475.
        1931725.       13871025.      1931423.02     13870345.54
#Sta/Elev= 30
  4600.3 1642.08  4687.7 1638.67  4811.4 1628.66    4829 1627.12    4880 1629.47
  4921.3 1619.84    4967 1613.53    5000 1612.78  5009.1 1610.39    5010 1609.89
  5046.2 1610.39  5073.1 1611.57  5093.6 1615.43    5151 1614.82  5182.2 1622.45
  5208.1    1621  5256.1 1630.15  5311.9 1630.58  5336.8 1626.66  5384.1 1634.08
  5417.4 1634.79  5441.9 1635.06  5598.3 1637.47    5745 1640.94  5854.2 1644.76
  5963.4 1649.02  6014.4 1650.41  6121.1 1659.04    6218  1676.8  6236.3  1678.5
#Mann= 12 ,-1 , 0
  4600.3     .07       0  4811.4    .035       0  4921.3      .1       0
  5009.1     .05       0  5046.2      .1       0  5417.4     .07       0
  5441.9      .1       0  5598.3     .07       0    5745      .1       0
  5854.2    .035       0  5963.4     .07       0  6121.1    .035       0
Bank Sta=5009.1,5046.2
XS Rating Curve= 0 ,0
Exp/Cntr=0.3,0.1

Type RM Length L Ch R = 1 ,50022   ,567,567,567
BEGIN DESCRIPTION:
Verde Creek 86.0
END DESCRIPTION:
XS GIS Cut Line= 4
      1932285.88     13872019.14        1932425.       13871575.
       1932416.8     13870944.94      1932411.38     13870528.31
#Sta/Elev= 30
  4543.2 1643.89  4773.8 1636.04  4798.2 1635.83  4808.2 1633.52  4855.3 1633.29
  4873.3 1630.19  4886.8 1625.86  4918.2  1610.6  4955.9 1612.53  4961.8 1611.08
    4962 1607.18  4962.9 1606.68  4999.2 1607.18  5036.3 1613.44  5054.3  1612.5
  5090.3 1614.43  5159.4 1622.95  5177.4 1620.48  5186.4 1625.35  5252.4 1632.27
  5370.3 1631.26  5516.4 1631.16  5672.4 1633.67  5837.4 1640.11  5909.4 1650.67
  5933.4 1661.39  5951.4 1661.96  5977.9  1674.5  6002.4 1682.93  6055.4 1693.55
#Mann= 7 ,-1 , 0
  4543.2     .07       0  4773.8    .035       0  4873.3      .1       0
    4962     .05       0  4999.2      .1       0  5370.3    .035       0
  5977.9     .07       0
Bank Sta=4962,4999.2
XS Rating Curve= 0 ,0
Exp/Cntr=0.3,0.1

Type RM Length L Ch R = 1 ,49455   ,518,518,518
BEGIN DESCRIPTION:
Verde Creek 85.0
END DESCRIPTION:
XS GIS Cut Line= 4
        1932975.     13872024.97        1932975.       13871625.
      1932918.48     13871164.08      1932850.47     13870609.48
#Sta/Elev= 30
  4604.6 1641.96  4611.5 1641.74  4709.9 1638.06  4731.3 1637.62  4811.8 1631.73
  4848.3  1626.6  4860.3 1623.24  4872.3 1617.07  4883.9  1612.6  4899.3    1609
  4911.3 1610.36  4952.9 1609.61  4961.6 1606.07  4962.6 1605.57  4998.9 1606.07
  5007.3 1608.57  5028.5 1611.66  5043.6 1610.58  5058.7 1612.07  5070.8 1614.76
  5076.8 1614.82  5134.3 1624.16  5204.1 1628.13  5218.9 1629.05  5224.9 1628.25
  5303.6 1627.92  5651.1  1631.9  5817.3 1632.67  5944.3 1636.13  6027.7  1640.6
#Mann= 8 ,-1 , 0
  4604.6      .1       0  4611.5     .07       0  4709.9    .035       0
  4811.8      .1       0  4961.6     .05       0  4998.9      .1       0
  5204.1     .07       0  5303.6    .035       0
Bank Sta=4961.6,4998.9
XS Rating Curve= 0 ,0
Exp/Cntr=0.3,0.1

Type RM Length L Ch R = 1 ,48937   ,626,626,626
BEGIN DESCRIPTION:
Verde Creek 84.0
END DESCRIPTION:
XS GIS Cut Line= 5
      1932741.98     13872262.84      1933408.11     13871863.23
      1933463.98     13871742.38        1933375.       13871075.
      1933324.62     13870697.17
#Sta/Elev= 30
  4144.5 1647.86  4246.9 1647.01  4320.8 1646.55  4555.2 1642.58  4589.3 1639.98
  4631.6 1639.67    4684 1636.55  4713.2 1638.11  4741.1 1636.95  4769.1 1637.77
  4791.8 1635.88  4818.1 1631.63  4863.6 1628.18  4905.6 1614.87  4938.9  1607.5
  4951.9 1606.52  4968.6 1607.14  4970.6 1604.37  4971.5 1603.87  5007.9 1604.37
    5038 1608.63    5103 1611.88  5142.3 1617.94  5172.6 1621.09  5246.2 1626.64
  5257.8 1626.64  5305.7 1625.86  5370.4 1627.16  6026.1 1630.95  6108.9 1632.71
#Mann= 11 ,-1 , 0
  4144.5      .1       0  4246.9     .07       0  4320.8      .1       0
  4555.2     .07       0  4589.3    .035       0  4791.8     .07       0
  4951.9      .1       0  4970.6     .05       0  5007.9      .1       0
  5257.8     .07       0  5370.4    .035       0
Bank Sta=4970.6,5007.9
XS Rating Curve= 0 ,0
Exp/Cntr=0.3,0.1

Type RM Length L Ch R = 1 ,48311   ,544,544,544
BEGIN DESCRIPTION:
Verde Creek 83.0
END DESCRIPTION:
XS GIS Cut Line= 4
      1933623.42     13872818.42        1934025.       13871925.
        1933925.       13871225.      1933863.84     13870796.88
#Sta/Elev= 30
  4015.5 1651.07  4015.8 1651.07  4077.8 1650.97  4096.8 1649.95  4114.2 1646.04
  4165.9 1639.14  4196.5 1637.87  4452.6  1630.8  4631.6 1628.66  4752.1 1627.08
    4850 1627.09  4869.7 1623.82  4890.3 1623.85  4902.6 1622.22  4928.9 1613.58
  4958.5 1606.13  4968.4 1604.69  4984.9  1605.6  4990.9 1603.21  4991.9 1602.71
  5028.9 1603.21  5040.1 1603.33  5049.3 1605.63  5066.5 1605.87  5107.4 1608.96
    5148 1614.34  5261.4 1622.91  5356.3 1623.57  5697.7 1628.03  6134.6 1629.01
#Mann= 11 ,-1 , 0
  4015.5     .07       0  4015.8      .1       0  4114.2    .035       0
  4631.6     .07       0  4752.1    .035       0  4890.3     .07       0
  4990.9     .05       0  5028.9     .07       0  5066.5      .1       0
    5148     .07       0  5356.3    .035       0
Bank Sta=4990.9,5028.9
XS Rating Curve= 0 ,0
Exp/Cntr=0.3,0.1

Type RM Length L Ch R = 1 ,47767   ,548,548,548
BEGIN DESCRIPTION:
Verde Creek 82.0
END DESCRIPTION:
XS GIS Cut Line= 4
        1934025.     13872774.99        1934525.       13871975.
        1934375.       13871275.       1934289.4     13870875.55
#Sta/Elev= 30
  4051.5  1649.4  4091.9 1646.37  4152.7 1636.39  4205.7  1633.4  4285.8 1629.76
    4392 1627.07  4535.1 1625.15  4774.5 1624.55    4820 1625.72  4834.2 1622.19
    4866 1622.71  4888.3 1618.39    4898 1617.69  4911.2 1615.52  4922.6 1609.06
  4933.8 1605.96  4940.3 1604.53  4955.2 1604.38  4967.3 1602.03  4968.3 1601.53
  5005.4 1602.03  5033.5  1603.7  5042.7 1606.53  5082.6 1606.75  5201.7 1615.53
  5204.8 1615.75  5251.3 1619.48  5309.6 1620.04  5407.8 1624.78  6119.3 1630.48
#Mann= 10 ,-1 , 0
  4051.5    .035       0  4091.9      .1       0  4205.7     .07       0
  4774.5    .035       0  4888.3     .07       0    4898      .1       0
  4967.3     .05       0  5005.4      .1       0  5201.7     .07       0
  5204.8    .035       0
Bank Sta=4967.3,5005.4
XS Rating Curve= 0 ,0
Exp/Cntr=0.3,0.1

Type RM Length L Ch R = 1 ,47219   ,180,180,180
BEGIN DESCRIPTION:
Verde Creek 81.0
END DESCRIPTION:
XS GIS Cut Line= 3
      1934897.32     13872903.25        1934975.       13872125.
      1934981.25     13871329.54
#Sta/Elev= 30
  4217.9 1629.23  4299.3 1629.57  4353.7 1628.23  4383.7 1626.27  4413.8 1622.12
  4459.1 1619.98  4507.3 1619.25  4516.3 1618.06  4546.5 1618.39  4585.7 1617.27
  4612.9  1618.9  4649.4 1618.21  4787.7  1615.7  4832.9 1611.83    4860 1608.15
  4917.5 1605.79    4951 1606.06  4962.6 1604.19  4995.1 1602.81  4996.1 1602.31
  5037.4 1602.81  5037.7 1606.96  5040.7  1607.4  5085.7 1609.16  5154.7 1616.85
  5220.7  1622.7  5264.2 1624.32  5448.6 1625.15    5732 1626.83  5795.5 1627.49
#Mann= 7 ,-1 , 0
  4217.9    .035       0  4353.7      .1       0  4649.4    .035       0
  4995.1    .035       0  5037.4    .035       0  5448.6     .07       0
    5732    .035       0
Bank Sta=4995.1,5037.4
XS Rating Curve= 0 ,0
Exp/Cntr=0.3,0.1

Type RM Length L Ch R = 1 ,47039   ,335,335,335
BEGIN DESCRIPTION:
Verde Creek 80.1
END DESCRIPTION:
XS GIS Cut Line= 3
      1935080.92     13872935.33      1935128.51     13872418.92
      1935154.35     13871382.34
#Sta/Elev= 30
    4248 1629.65  4311.5 1626.31  4602.4 1620.34  4650.8 1621.82  4677.9 1621.06
  4701.9 1615.75  4726.1 1613.19  4774.3  1609.8    4804 1608.77  4852.3 1606.27
  4945.3 1604.38  4949.8 1603.45  4977.8 1602.49  4978.8 1601.99  5020.2 1602.49
  5020.3 1604.15  5031.8 1605.51  5071.3 1607.03    5099 1610.95  5122.1 1614.59
  5140.4 1616.17  5197.4  1618.6    5269 1620.14  5512.5 1623.19  5536.5 1622.18
  5551.5 1623.61  5587.5 1624.66  5614.5 1623.07  5626.5 1624.08  5803.5 1624.93
#Mann= 6 ,-1 , 0
    4248    .035       0  4311.5    .063       0    4804    .035       0
  4977.8    .035       0  5020.2    .035       0    5099    .063       0
Bank Sta=4977.8,5020.2
XS Rating Curve= 0 ,0
Exp/Cntr=0.3,0.1

Type RM Length L Ch R = 1 ,46704   ,531,531,531
BEGIN DESCRIPTION:
Verde Creek 80.0
END DESCRIPTION:
XS GIS Cut Line= 3
      1935148.15      13873569.6        1935425.       13872325.
        1936225.       13871525.
#Sta/Elev= 30
  3729.6 1643.23  3790.9 1640.71  4349.4 1626.68  4396.8  1626.8  4510.6  1622.5
  4593.5 1622.16  4710.3 1615.69  4759.5  1615.3  4765.6    1613  4808.7 1609.94
  4851.7 1603.37  4906.2 1602.04  4947.9 1602.81  5001.4 1600.12  5002.4 1599.62
  5043.8 1600.12    5099 1611.34  5173.2 1619.09  5199.4 1619.43  5320.6 1619.67
  5326.1 1619.67  5619.2 1620.02  5688.7 1619.73  5718.3 1621.19  5752.3 1618.89
    5782 1621.62  6049.7 1631.55  6104.5 1638.21    6128  1639.2    6136 1639.17
#Mann= 12 ,-1 , 0
  3729.6    .035       0  3790.9     .07       0  4349.4    .035       0
  4906.2      .1       0  5001.4     .05       0  5043.8      .1       0
  5199.4     .07       0  5320.6    .035       0  5326.1     .07       0
  5619.2    .035       0  6049.7      .1       0    6128    .035       0
Bank Sta=5001.4,5043.8
XS Rating Curve= 0 ,0
Exp/Cntr=0.3,0.1

Type RM Length L Ch R = 1 ,46173   ,572,572,572
BEGIN DESCRIPTION:
Verde Creek 79.0
END DESCRIPTION:
XS GIS Cut Line= 3
      1935487.19     13873723.78      1935870.69     13872570.65
      1936316.26     13871501.83
#Sta/Elev= 30
  3784.7 1642.87  3900.8 1636.05  4104.9 1628.85  4479.8 1622.73  4676.7  1619.6
  4750.5  1621.2  4804.3 1620.17  4816.9 1617.15  4839.1 1608.19  4861.2 1604.58
  4908.6 1601.26  4967.4 1600.31  4978.5 1597.16  4981.3 1593.96  4982.3 1593.46
  5023.8 1593.96  5029.6 1600.01  5077.4 1602.32  5107.6 1605.35  5155.4 1613.23
    5177 1614.39  5702.4 1619.95  5742.6 1617.64  5757.6 1620.55  5812.9 1621.61
  5885.2 1625.79  5949.4 1630.95  6076.8 1637.92  6114.4 1640.13  6157.9 1642.65
#Mann= 10 ,-1 , 0
  3784.7    .035       0  3900.8     .07       0  4479.8    .035       0
  4967.4      .1       0  4981.3     .05       0  5023.8      .1       0
    5177    .035       0  5885.2      .1       0  6076.8    .035       0
  6114.4      .1       0
Bank Sta=4981.3,5023.8
XS Rating Curve= 0 ,0
Exp/Cntr=0.3,0.1

Type RM Length L Ch R = 1 ,45601   ,564,564,564
BEGIN DESCRIPTION:
Verde Creek 78.0
END DESCRIPTION:
XS GIS Cut Line= 3
      1935812.11     13873926.49        1936375.       13872775.
      1936384.95     13871633.95
#Sta/Elev= 30
  3718.3  1640.7  3851.2 1631.58  3952.1 1628.76  3990.2 1625.64  4060.6 1623.48
  4279.6 1618.59  4702.5 1619.24  4740.9 1620.17  4788.7 1618.44  4823.8 1602.67
  4848.8 1601.41  4954.1 1599.84  4967.4 1597.92  4968.8 1592.66  4969.8 1592.16
  5011.3 1592.66  5024.7 1597.51  5131.7 1600.98  5235.2 1607.84  5354.7 1608.03
  5422.8 1611.92  5639.5 1615.84  5746.6 1618.61  5780.8 1616.25  5795.8 1619.15
  5813.8 1620.17  5928.9 1623.31  6005.8 1626.99  6077.2 1634.39  6141.1 1638.92
#Mann= 11 ,-1 , 0
  3718.3    .035       0  4060.6     .05       0  4702.5    .035       0
  4740.9     .05       0  4848.8      .1       0  4968.8     .05       0
  5011.3      .1       0  5131.7     .07       0  5639.5    .035       0
  5928.9      .1       0  6077.2    .035       0
Bank Sta=4968.8,5011.3
XS Rating Curve= 0 ,0
Exp/Cntr=0.3,0.1

Type RM Length L Ch R = 1 ,45037   ,553,553,553
BEGIN DESCRIPTION:
Verde Creek 77.0
END DESCRIPTION:
XS GIS Cut Line= 3
      1936004.31     13874336.49        1936875.       13872775.
        1937125.     13871974.99
#Sta/Elev= 30
  3219.9 1653.09    3320  1645.3  3459.4 1635.43  3600.3 1628.98  3746.6 1622.72
  3967.8 1617.84  4624.6 1618.01  4834.7 1616.99    4858 1616.38  4879.2 1607.57
  4895.2 1598.18  4920.7 1596.22    4922 1591.38    4923 1590.88  4964.5 1591.38
  5154.3 1601.05  5230.7 1601.28  5263.1 1598.96  5303.9 1601.45  5344.8  1607.9
  5460.5 1614.69  5492.5 1614.96  5511.4 1612.73  5539.7 1617.31    5647 1621.78
    5700 1625.72  5731.4 1632.31  5794.3 1638.86  5816.3 1644.52  5845.9 1646.88
#Mann= 11 ,-1 , 0
  3219.9     .07       0    3320    .035       0  3600.3     .05       0
  4624.6    .035       0  4834.7      .1       0  4879.2      .1       0
    4922     .05       0  4964.5      .1       0  5154.3     .07       0
  5460.5    .035       0    5647     .07       0
Bank Sta=4922,4964.5
XS Rating Curve= 0 ,0
Exp/Cntr=0.3,0.1

Type RM Length L Ch R = 1 ,44484   ,548,548,548
BEGIN DESCRIPTION:
Verde Creek 76.0
END DESCRIPTION:
XS GIS Cut Line= 3
      1936324.51     13874081.52        1937325.       13872675.
      1937525.02     13872324.97
#Sta/Elev= 30
  3273.9 1628.41  3472.5 1620.87  3795.7 1615.61  4506.4 1616.14  4679.3 1616.08
  4698.3 1614.22  4730.9 1615.58  4798.4 1610.57  4831.7 1607.16  4874.4 1596.83
  4914.3 1592.26  4956.5 1595.21  4970.2 1594.32  4972.7  1590.3  4973.7  1589.8
  5015.5  1590.3  5030.5  1592.8  5037.6 1595.32  5061.8 1598.85  5111.6 1609.35
  5141.8 1610.62  5189.7 1613.16  5217.3 1611.07    5238 1618.47  5296.3 1621.38
  5310.6  1624.3  5326.6  1630.3  5345.2 1637.12  5355.5 1639.29  5403.1  1642.4
#Mann= 9 ,-1 , 0
  3273.9     .05       0  4506.4    .035       0  4798.4     .07       0
  4914.3    .035       0  4972.7    .035       0  5015.5    .035       0
  5030.5      .1       0  5141.8    .035       0  5326.6     .07       0
Bank Sta=4972.7,5015.5
XS Rating Curve= 0 ,0
Exp/Cntr=0.3,0.1

Type RM Length L Ch R = 1 ,43936   ,545,545,545
BEGIN DESCRIPTION:
Verde Creek 75.0
END DESCRIPTION:
XS GIS Cut Line= 4
      1936031.37     13874468.43      1937444.88     13873275.61
        1937775.       13872925.      1938575.01     13872124.99
#Sta/Elev= 30
  2669.1  1661.4  2732.2 1656.33  2780.1 1650.49  3146.1  1630.3  3514.4 1618.34
  3878.5 1614.17  4694.6 1612.78  4735.4 1611.17  4837.7 1604.29  4884.2 1598.17
    4957 1593.91    5008 1590.71    5009 1590.21  5050.8 1590.71  5094.6 1592.81
  5117.8 1597.38  5213.4 1610.37  5234.6 1610.04  5247.3 1604.61    5267 1601.52
  5339.1 1602.39  5677.1 1631.17  5746.4 1636.96  5777.6 1645.18  5840.2 1652.81
  5945.8 1667.41  5971.2 1666.91  6036.3 1677.14  6038.6  1677.3  6131.6 1686.59
#Mann= 15 ,-1 , 0
  2669.1    .035       0  2732.2     .07       0  2780.1    .035       0
  3146.1     .05       0  4694.6    .035       0  4735.4     .05       0
  4884.2     .07       0    4957      .1       0    5008     .05       0
  5050.8      .1       0  5117.8    .035       0  5677.1     .07       0
  5840.2    .035       0  6036.3     .07       0  6038.6    .035       0
Bank Sta=5008,5050.8
XS Rating Curve= 0 ,0
Exp/Cntr=0.3,0.1

Type RM Length L Ch R = 1 ,43391   ,537,537,537
BEGIN DESCRIPTION:
Verde Creek 74.0
END DESCRIPTION:
XS GIS Cut Line= 4
      1936096.18      13874544.2        1937775.       13873425.
        1938225.       13873125.      1938975.01       13872825.
#Sta/Elev= 30
  2434.1 1664.04  2528.2 1655.98  2768.2 1639.17  2841.9 1635.05  3031.2 1628.47
  3354.5 1618.34    4347 1610.02  4498.9 1610.97  4748.6    1601  4821.9 1594.58
    4871 1590.87  4917.9 1592.11  4986.9 1586.49  4987.9 1585.99  5029.8 1586.49
    5091  1596.6  5123.7 1598.15  5173.1 1611.07    5216 1610.48    5241 1604.05
  5279.8 1613.11  5346.3 1619.17  5438.1 1628.24  5463.9 1628.02  5506.8 1634.78
  5564.1 1642.13  5641.4  1662.1  5678.1 1665.66  5713.7 1674.83  5800.4 1686.87
#Mann= 15 ,-1 , 0
  2434.1     .07       0  2528.2    .035       0  2768.2     .05       0
  2841.9    .035       0  3031.2     .05       0    4347    .035       0
  4748.6     .05       0  4821.9     .07       0  4917.9      .1       0
  4986.9     .05       0  5029.8      .1       0    5091    .035       0
  5346.3     .07       0  5506.8    .035       0  5641.4     .07       0
Bank Sta=4986.9,5029.8
XS Rating Curve= 0 ,0
Exp/Cntr=0.3,0.1

Type RM Length L Ch R = 1 ,42854   ,539,539,539
BEGIN DESCRIPTION:
Verde Creek 73.0
END DESCRIPTION:
XS GIS Cut Line= 4
      1937405.01     13875552.12        1938325.       13873975.
        1938675.       13873375.      1938875.01     13873024.98
#Sta/Elev= 30
  2479.3 1629.11  2783.9 1626.86  3429.1 1618.63  3652.8  1615.6  3746.7 1615.17
    3761 1615.21  4320.3  1608.5  4563.5 1599.11  4712.7 1597.17  4820.7 1589.77
  4879.4  1588.4  4923.2 1590.74  4957.3 1588.17  4965.9 1586.57  4968.6  1582.8
  4969.6  1582.3  5011.8  1582.8  5014.4 1585.47  5038.6 1588.55  5048.4 1596.55
  5067.2 1604.97  5128.4 1611.29  5173.4 1613.13  5204.4 1619.81  5218.3 1619.77
  5254.7 1632.17  5283.5 1634.82  5315.4 1641.31  5363.7 1658.08  5402.9 1662.88
#Mann= 10 ,-1 , 0
  2479.3     .07       0  2783.9    .035       0  3429.1     .07       0
  3652.8    .035       0  3746.7     .07       0    3761    .035       0
  4820.7     .07       0  4968.6    .035       0  5011.8      .1       0
  5283.5     .07       0
Bank Sta=4968.6,5011.8
XS Rating Curve= 0 ,0
Exp/Cntr=0.3,0.1

Type RM Length L Ch R = 1 ,42315   ,559,559,559
BEGIN DESCRIPTION:
Verde Creek 72.0
END DESCRIPTION:
XS GIS Cut Line= 4
      1937428.81     13875570.55        1938625.       13874175.
        1938925.       13873825.      1939274.99     13873025.03
#Sta/Elev= 30
    2701 1630.02    2917 1628.16    3294 1624.89  3795.1 1614.92  4116.1  1612.1
  4462.3 1607.59  4523.2 1606.74    4686 1601.45  4748.1 1595.14  4883.7 1592.62
    4986 1581.23    4987 1580.73  5029.3 1581.23  5030.6 1587.07  5073.2 1587.94
  5097.4 1592.98    5112 1596.39  5141.9  1596.2  5153.4 1601.01  5187.8  1606.6
  5221.4 1605.76  5233.6 1601.64  5259.3 1606.89  5482.5 1616.23  5549.9 1623.72
  5633.1 1641.09  5685.5 1660.31  5770.6 1668.32  5803.4 1677.01  5873.2 1686.21
#Mann= 14 ,-1 , 0
    2701     .07       0    2917    .035       0  3795.1     .07       0
  4116.1    .035       0  4462.3     .07       0  4523.2    .035       0
    4686     .07       0  4883.7      .1       0    4986     .05       0
  5029.3      .1       0  5097.4    .035       0  5153.4      .1       0
  5259.3    .035       0  5549.9     .07       0
Bank Sta=4986,5029.3
XS Rating Curve= 0 ,0
Exp/Cntr=0.3,0.1

Type RM Length L Ch R = 1 ,41756   ,541,541,541
BEGIN DESCRIPTION:
Verde Creek 71.0
END DESCRIPTION:
XS GIS Cut Line= 4
      1937897.87     13875663.29        1939075.       13874675.
        1939225.       13874275.      1939643.64     13873161.49
#Sta/Elev= 30
  3031.5 1629.85  3138.4 1627.12  3151.1  1626.8  3471.9 1618.76  3546.2 1616.37
  3732.8 1613.19  4419.6 1608.95  4456.3  1609.3  4572.6  1608.6  4676.5 1605.01
    4875 1600.56    4988 1582.38  4991.2 1580.21  4992.2 1579.71  5034.5 1580.21
  5067.3 1584.92  5115.4 1585.68  5195.7 1598.19  5299.6 1603.91  5323.4  1604.1
  5373.4  1604.5  5397.4 1608.09  5458.3    1605  5615.3 1609.99  5803.9 1616.17
    5891 1621.66  5952.4 1633.82  5990.3 1642.12  6051.3 1664.64  6185.3 1685.57
#Mann= 19 ,-1 , 0
  3031.5     .07       0  3138.4    .035       0  3151.1     .07       0
  3471.9    .035       0  3546.2     .07       0  3732.8    .045       0
  4419.6     .07       0  4456.3    .045       0  4572.6     .07       0
  4676.5    .035       0    4988      .1       0  4991.2     .05       0
  5034.5      .1       0  5195.7    .035       0  5299.6     .07       0
  5323.4    .035       0  5615.3     .07       0  5803.9    .035       0
  5952.4     .07       0
Bank Sta=4991.2,5034.5
XS Rating Curve= 0 ,0
Exp/Cntr=0.3,0.1

Type RM Length L Ch R = 1 ,41215   ,426,426,426
BEGIN DESCRIPTION:
Verde Creek 70.0
END DESCRIPTION:
XS GIS Cut Line= 4
      1937734.96     13875806.27        1939225.       13874875.
        1939625.       13874625.      1939877.89     13873474.69
#Sta/Elev= 30
  2775.6  1634.7  3183.2 1625.73  3487.5 1616.23  3618.7 1614.38  4013.3 1609.22
  4399.6 1608.06  4549.8 1607.99    4636 1602.98  4755.3 1598.63    4778 1599.11
  4845.9 1595.16  4873.9 1590.64  4890.3 1589.25  4924.8 1584.68  4981.4 1584.03
  4988.9 1579.73  4989.9 1579.23  5032.2 1579.73  5050.5 1582.42  5078.7 1581.82
  5161.8 1596.97  5231.7 1600.94  5297.7 1601.76    5373 1603.31  5397.6 1605.76
  5452.9 1601.97    5778 1610.25  6097.1 1617.48  6128.7 1618.63  6182.2 1629.73
#Mann= 12 ,-1 , 0
  2775.6     .07       0  3618.7    .045       0  4399.6     .07       0
    4636    .035       0  4755.3      .1       0  4873.9     .07       0
  4890.3      .1       0  4988.9     .05       0  5032.2      .1       0
  5297.7    .035       0    5778     .07       0  6097.1    .035       0
Bank Sta=4988.9,5032.2
XS Rating Curve= 0 ,0
Exp/Cntr=0.3,0.1

Type RM Length L Ch R = 1 ,40789   ,648,648,648
BEGIN DESCRIPTION:
Verde Creek 69.0
END DESCRIPTION:
XS GIS Cut Line= 4
      1938574.33     13876311.46      1939759.93     13875039.38
      1939964.79     13874858.25      1940114.17      13873371.8
#Sta/Elev= 30
  3109.1 1638.36  3639.8 1624.95  3745.4 1620.83  3754.7 1622.31  3847.9 1617.51
  4512.3 1600.36  4615.7  1600.9    4655 1599.88  4757.7 1593.03  4799.3 1591.63
  4866.1 1581.82  4901.7 1580.87  4956.6 1578.03  4957.6 1577.53  4999.9 1578.03
  5026.3 1587.61  5070.5 1599.03  5182.1 1600.49  5452.4 1601.18  5515.7 1603.72
    5570 1600.01  5591.1 1602.13  5722.5 1603.33  6402.2 1610.98  6453.4 1612.32
  6522.7 1619.61  6540.8 1619.53    6562 1626.27  6589.1 1637.21  6615.4 1641.89
#Mann= 12 ,-1 , 0
  3109.1     .07       0  3639.8    .035       0  4615.7     .07       0
    4655    .035       0  4757.7     .07       0  4901.7      .1       0
  4956.6     .05       0  4999.9      .1       0  5182.1    .035       0
  5722.5     .07       0  6402.2    .035       0    6562      .1       0
Bank Sta=4956.6,4999.9
XS Rating Curve= 0 ,0
Exp/Cntr=0.3,0.1

Type RM Length L Ch R = 1 ,40141   ,577,577,577
BEGIN DESCRIPTION:
Verde Creek 68.0
END DESCRIPTION:
XS GIS Cut Line= 5
      1938527.32     13876416.52        1939825.       13875675.
        1940175.       13875475.      1940355.74     13875037.21
      1940197.52     13873344.43
#Sta/Elev= 30
  3098.6 1641.37  3359.4 1635.19  3390.3 1634.46  3502.9 1631.21  3755.9 1625.77
  3806.9 1624.64  4053.6 1614.63  4453.6 1606.88  4771.1 1601.63  4883.5 1596.48
  4922.7 1585.92  4927.9 1577.64  4928.9 1577.14    4972 1577.64  5008.6 1577.71
  5072.1 1578.95  5153.2 1593.34  5288.4 1598.53  5292.3 1598.72  5500.5  1597.8
  5733.2 1598.76  5847.8 1601.53    5899 1597.58  5911.1 1600.71  6228.4 1604.11
  6915.1 1611.31    7038 1615.12  7071.1 1620.63  7086.2 1626.05  7170.1 1648.11
#Mann= 18 ,-1 , 0
  3098.6     .07       0  3359.4    .035       0  3390.3     .07       0
  3502.9    .035       0  3755.9     .07       0  3806.9    .035       0
  4453.6     .07       0  4771.1      .1       0  4927.9     .05       0
    4972      .1       0  5008.6      .1       0  5288.4     .07       0
  5292.3    .035       0  5500.5      .1       0  5733.2    .035       0
  6228.4     .07       0  6915.1    .035       0  7086.2      .1       0
Bank Sta=4927.9,4972
XS Rating Curve= 0 ,0
Exp/Cntr=0.3,0.1

Type RM Length L Ch R = 1 ,39564   ,560,560,560
BEGIN DESCRIPTION:
Verde Creek 67.0
END DESCRIPTION:
XS GIS Cut Line= 4
      1940435.06     13877094.55        1940575.       13875975.
        1940625.       13875575.      1940334.04     13873612.93
#Sta/Elev= 30
  3472.9 1619.82  3492.6  1619.2  3494.6 1640.68  3497.7    1619  4719.1 1601.07
  4782.6 1597.81    4816 1587.57    4843 1586.32  4855.1 1582.73  4891.4 1576.92
  4906.5 1575.76  4939.8  1578.1  4953.8 1571.29  4954.8 1570.79  4998.4 1571.29
  5003.3 1572.33  5018.4  1582.1  5053.1 1587.15  5076.1 1590.05  5177.8 1595.16
  5310.9    1596  5372.8 1596.05  5494.2 1595.35  5646.2 1597.13    5807 1600.29
  5858.5 1596.66  5879.8 1600.11  6375.9 1606.17  6870.3 1607.85  6987.8 1609.91
#Mann= 8 ,-1 , 0
  3472.9     .07       0  4953.8     .05       0  4998.4     .07       0
  5177.8     .07       0  5310.9    .035       0  5372.8     .07       0
  5646.2    .035       0  6375.9     .07       0
Bank Sta=4953.8,4998.4
XS Rating Curve= 0 ,0
Exp/Cntr=0.3,0.1

Type RM Length L Ch R = 1 ,39004   ,507,507,507
BEGIN DESCRIPTION:
Verde Creek 66.0
END DESCRIPTION:
XS GIS Cut Line= 3
        1940875.       13876175.        1941075.       13875825.
      1942250.54      13874337.3
#Sta/Elev= 30
  4596.9 1602.66  4765.1 1597.78  4868.7 1591.84  4941.3 1584.53  4969.6 1577.63
  4972.7 1571.94  4973.7 1571.44  5017.3 1571.94  5017.5 1573.32  5057.4 1578.88
  5080.3 1576.63  5114.7 1576.69  5183.6 1583.44  5228.9 1582.31  5280.5 1577.98
  5294.4  1573.6  5305.7 1574.91  5334.7 1589.79  5354.1 1593.83    5495 1595.95
  5686.2 1596.01  5780.7  1596.9  6422.9 1602.35  6517.4 1608.45  6544.4 1608.38
  6575.3 1611.93    6617 1622.43    6738 1630.51  6788.6 1637.42  6896.1 1643.55
#Mann= 9 ,-1 , 0
  4596.9      .1       0  4972.7     .05       0  5017.3      .1       0
  5280.5    .035       0    5495     .07       0  5686.2    .035       0
  5780.7     .07       0  6517.4    .035       0  6788.6     .07       0
Bank Sta=4972.7,5017.3
XS Rating Curve= 0 ,0
Exp/Cntr=0.3,0.1

Type RM Length L Ch R = 1 ,38497   ,604,604,604
BEGIN DESCRIPTION:
Verde Creek 65.0
END DESCRIPTION:
XS GIS Cut Line= 3
      1941324.99     13876525.03      1941458.41       13876129.
        1942325.     13874574.99
#Sta/Elev= 30
  4567.2 1599.66  4699.3 1595.82  4834.2 1587.12  4927.6 1577.59  4970.3  1576.6
  4972.8 1572.48  4973.8 1571.98  5020.3 1572.48  5055.1 1577.42  5127.1 1576.86
  5156.7 1580.05  5206.1 1591.16  5297.6 1592.39  5322.9  1591.3  5366.9 1593.71
  5537.1  1594.5  5862.4 1594.45  6039.7 1596.85  6151.5 1599.72  6184.1 1602.97
  6246.9 1602.68  6386.4 1606.82  6416.4 1607.33  6540.4  1616.5  6562.9  1618.3
  6604.1  1626.7  6645.3 1630.26  6683.1  1638.7  6741.5 1641.98  6764.4 1645.38
#Mann= 10 ,-1 , 0
  4567.2      .1       0  4699.3     .07       0  4972.8     .05       0
  5020.3     .07       0  5156.7    .035       0  5366.9     .07       0
  5537.1    .035       0  6039.7     .07       0  6386.4    .035       0
  6540.4     .07       0
Bank Sta=4972.8,5020.3
XS Rating Curve= 0 ,0
Exp/Cntr=0.3,0.1

Type RM Length L Ch R = 1 ,37893   ,588,588,588
BEGIN DESCRIPTION:
Verde Creek 64.0
END DESCRIPTION:
XS GIS Cut Line= 3
        1941375.       13876575.        1941775.       13876525.
      1942693.61     13875024.24
#Sta/Elev= 30
  4591.3 1599.15  4663.6 1597.76  4769.1 1590.82    4863 1584.42  4897.2 1581.34
  4948.6 1574.51  4966.7 1573.53  4969.7 1572.44  4970.2 1568.54  4971.2 1568.04
  5017.7 1568.54  5022.2 1570.39  5049.3 1570.42    5069 1573.58    5088 1570.44
  5104.7 1572.19  5197.7 1581.91  5224.2 1587.35  5273.5 1590.01  5319.2 1587.87
  5336.8 1590.64  5383.3 1590.99  5437.9 1591.47  5758.4 1592.73  5931.2 1592.07
  6148.5 1593.73  6320.9 1598.93  6546.7 1611.74  6641.7 1617.07    6754 1627.93
#Mann= 11 ,-1 , 0
  4591.3      .1       0  4663.6     .07       0  4769.1      .1       0
    4863     .07       0  4970.2     .05       0  5017.7     .07       0
    5088      .1       0  5104.7    .035       0  5383.3     .07       0
  5437.9    .035       0  6546.7     .07       0
Bank Sta=4970.2,5017.7
XS Rating Curve= 0 ,0
Exp/Cntr=0.3,0.1
