--- BIG JOSHUA CREEK.prj (project) ---

Proj Title=BIG JOSHUA CREEK Base Level Engineering
Current Plan=p01
Default Exp/Contr=0.3,0.1
English Units
Geom File=g01
Flow File=f01
Plan File=p01
Y Axis Title=Elevation
X Axis Title(PF)=Main Channel Distance
X Axis Title(XS)=Station
BEGIN DESCRIPTION:
BIG JOSHUA CREEK
END DESCRIPTION:
DSS Export Rating Curves= 0
DSS Export Rating Curve Sorted= 0
DSS Export Volume Flow Curves= 0
DXF OffsetX= 0
DXF OffsetY= 0
DXF ScaleX= 1
DXF ScaleY= 10

--- BIG JOSHUA CREEK.p01 (plan) ---

Plan Title=Multiple Run
Short Identifier=Multiple
Geom File=g01
Flow File=f01
Subcritical Flow
K Sum by GR= 0
Std Step Tol= 0.01
Critical Tol= 0.01
Num of Std Step Trials= 20
Max Error Tol= 0.3
Flow Tol Ratio= 0.001
Split Flow NTrial= 30
Split Flow Tol= 0.02
Split Flow Ratio= 0.02
Log Output Level= 0
Friction Slope Method= 1
Unsteady Friction Slope Method= 2
Unsteady Bridges Friction Slope Method= 1
Parabolic Critical Depth
Global Vel Dist=  1 , 1 , 1
Global Log Level= 0
CheckData=True
Encroach Param= -1, 0, 0, 0
BEGIN DESCRIPTION:
Multiple Run
END DESCRIPTION:

--- BIG JOSHUA CREEK.f01 (steady flow) ---

Flow Title=Multiple
Program Version=4.10
Number of Profiles= 7
Profile Names=10-year,25-year,50-year,1pct_min,100-year,1pct_plu,500-year
River Rch & RM=BIG JOSHUA CREEK,Reach-1         ,70319
     301     468     616     394     787    1570    1267
River Rch & RM=BIG JOSHUA CREEK,Reach-1         ,69977
     663    1094    1495     993    1981    3953    3435
River Rch & RM=BIG JOSHUA CREEK,Reach-1         ,67218
    1011    1715    2387    1611    3215    6415    5768
River Rch & RM=BIG JOSHUA CREEK,Reach-1         ,65649
    1834    3222    4589    3164    6312   12595   11826
River Rch & RM=BIG JOSHUA CREEK,Reach-1         ,64481
    2060    3621    5159    3554    7091   14148   13267
River Rch & RM=BIG JOSHUA CREEK,Reach-1         ,59333
    3352    6002    8653    6021   12014   23971   22944
River Rch & RM=BIG JOSHUA CREEK,Reach-1         ,54329
    3452    6186    8924    6212   12394   24729   23684
River Rch & RM=BIG JOSHUA CREEK,Reach-1         ,52994
    3720    6670    9624    6697   13363   26662   25527
River Rch & RM=BIG JOSHUA CREEK,Reach-1         ,48796
    3942    7085   10239    7136   14238   28408   27278
River Rch & RM=BIG JOSHUA CREEK,Reach-1         ,47375
    4022    7225   10439    7272   14509   28950   27773
River Rch & RM=BIG JOSHUA CREEK,Reach-1         ,43722
    4122    7411   10713    7466   14898   29724   28544
River Rch & RM=BIG JOSHUA CREEK,Reach-1         ,43265
    4183    7513   10854    7558   15080   30089   28844
River Rch & RM=BIG JOSHUA CREEK,Reach-1         ,38321
    4827    8723   12652    8843   17643   35203   33997
River Rch & RM=BIG JOSHUA CREEK,Reach-1         ,37853
    5125    9274   13464    9417   18789   37488   36252
River Rch & RM=BIG JOSHUA CREEK,Reach-1         ,34138
    5407    9801   14243    9971   19894   39693   38454
River Rch & RM=BIG JOSHUA CREEK,Reach-1         ,31335
    5699   10343   15045   10540   21030   41960   40707
River Rch & RM=BIG JOSHUA CREEK,Reach-1         ,27034
    5986   10878   15838   11104   22156   44206   42954
River Rch & RM=BIG JOSHUA CREEK,Reach-1         ,25397
    6054   10992   15993   11204   22355   44604   43273
River Rch & RM=BIG JOSHUA CREEK,Reach-1         ,19917
    6297   11439   16650   11667   23278   46445   45076
River Rch & RM=BIG JOSHUA CREEK,Reach-1         ,17700
    6503   11833   17242   12095   24132   48149   46830
River Rch & RM=BIG JOSHUA CREEK,Reach-1         ,15567
    7014   12788   18658   13103   26143   52162   50845
River Rch & RM=BIG JOSHUA CREEK,Reach-1         ,11053
    7233   13191   19251   13519   26975   53822   52469
River Rch & RM=BIG JOSHUA CREEK,Reach-1         ,7242
    7458   13608   19866   13955   27844   55556   54185
River Rch & RM=BIG JOSHUA CREEK,Reach-1         ,4982
    7531   13731   20036   14066   28066   55999   54555
Boundary for River Rch & Prof#=BIG JOSHUA CREEK,Reach-1         , 1
Up Type= 0
Dn Type= 3
Dn Slope=0.008
Boundary for River Rch & Prof#=BIG JOSHUA CREEK,Reach-1         , 2
Up Type= 0
Dn Type= 3
Dn Slope=0.008
Boundary for River Rch & Prof#=BIG JOSHUA CREEK,Reach-1         , 3
Up Type= 0
Dn Type= 3
Dn Slope=0.008
Boundary for River Rch & Prof#=BIG JOSHUA CREEK,Reach-1         , 4
Up Type= 0
Dn Type= 3
Dn Slope=0.008
Boundary for River Rch & Prof#=BIG JOSHUA CREEK,Reach-1         , 5
Up Type= 0
Dn Type= 3
Dn Slope=0.008
Boundary for River Rch & Prof#=BIG JOSHUA CREEK,Reach-1         , 6
Up Type= 0
Dn Type= 3
Dn Slope=0.008
Boundary for River Rch & Prof#=BIG JOSHUA CREEK,Reach-1         , 7
Up Type= 0
Dn Type= 3
Dn Slope=0.008
DSS Import GetInterval= 0
DSS Import GetPeak= 0
DSS Import FillOption= 0

--- BIG JOSHUA CREEK.g01 (geometry) ---

Geom Title=Existing Conditions
Program Version=4.10

River Reach=BIG JOSHUA CREEK,Reach-1
Reach XY= 30
        1995575.       13853575.        1995175.       13854425.
        1996825.       13856925.      1996685.65       13858985.
      1999369.83     13859730.41      2000872.69     13862169.18
      2002195.55     13862044.44      2002280.45     13863577.47
      2003180.44     13864572.83      2004208.37     13864108.29
      2005130.02     13866769.77      2006923.54     13866928.53
        2006675.       13867625.      2007817.24     13868068.83
      2007380.59     13869119.39      2009377.58     13868280.71
      2009718.65     13869117.57      2010961.37     13869361.79
      2011083.14     13870881.06      2012648.84     13871597.85
      2013664.95     13873363.88      2017477.67     13874530.42
      2019880.73      13876873.1      2021127.55     13875480.72
      2023821.58     13878917.21      2025219.02     13878427.17
      2025926.46     13879371.46      2032577.45     13880980.47
      2034238.69       13884088.        2035175.       13884075.

Type RM Length L Ch R = 1 ,70319   ,342,342,342
BEGIN DESCRIPTION:
BIG JOSHUA CREEK 131.0
END DESCRIPTION:
XS GIS Cut Line= 3
      1995285.26     13853524.28        1995575.       13853675.
       1995908.4     13853724.83
#Sta/Elev= 30
  4673.4 1961.14  4682.3 1961.47  4788.7 1954.81  4853.5 1950.71  4881.2  1947.7
  4903.3  1944.8  4919.8 1940.88  4925.4 1940.55  4941.9  1936.2  4947.6 1935.95
    4964 1927.65  4969.7 1926.51  4977.5 1921.29  4986.1 1913.86  4991.8 1912.64
  4995.2 1910.04  4995.4 1909.54  4999.2 1910.04  5000.3 1910.04  5010.1 1912.58
  5040.4 1928.83  5070.8 1934.72  5098.6 1937.79  5103.8 1941.34  5161.8 1945.53
    5173 1948.08  5232.1 1954.04  5237.2 1955.65  5293.2 1958.86  5337.1 1962.93
#Mann= 6 ,-1 , 0
  4673.4     .12       0  4788.7     .07       0  4995.2     .05       0
  4999.2     .07       0  5000.3     .12       0  5098.6     .07       0
Bank Sta=4995.2,4999.2
XS Rating Curve= 0 ,0
Exp/Cntr=0.3,0.1

Type RM Length L Ch R = 1 ,69977   ,724,724,724
BEGIN DESCRIPTION:
BIG JOSHUA CREEK 130.0
END DESCRIPTION:
XS GIS Cut Line= 4
      1995284.21     13853758.33        1995475.       13853975.
      1995615.83     13854014.69      1995860.17     13853984.66
#Sta/Elev= 30
  4711.3  1949.1  4716.8 1948.22  4745.3 1947.64    4787 1947.88  4886.6 1937.91
  4921.7 1929.55  4929.3 1926.34  4943.5 1922.81  4964.4  1918.8  4986.2 1910.86
  4992.9  1906.9  4996.7  1900.7  5002.6  1900.7  5008.4 1898.53  5008.6 1898.03
  5012.4 1898.53    5017 1906.39  5022.2  1912.1  5041.6 1923.42    5051 1927.93
  5062.3 1935.81  5083.1 1944.74  5090.2 1947.05  5103.9 1949.41  5129.4 1952.04
  5143.3 1954.33  5179.6 1957.64  5216.4  1959.3  5264.1 1963.22  5392.5 1963.09
#Mann= 5 ,-1 , 0
  4711.3     .07       0  5008.4     .05       0  5012.4     .07       0
  5179.6     .12       0  5216.4    .035       0
Bank Sta=5008.4,5012.4
XS Rating Curve= 0 ,0
Exp/Cntr=0.3,0.1

Type RM Length L Ch R = 1 ,69253   ,745,745,745
BEGIN DESCRIPTION:
BIG JOSHUA CREEK 129.0
END DESCRIPTION:
XS GIS Cut Line= 3
      1994775.59     13854640.03        1995225.       13854525.
       1995629.8     13854269.86
#Sta/Elev= 30
  4536.1 1951.37    4604  1947.7    4649 1945.14    4680 1939.88  4729.9 1937.55
    4809 1929.09  4859.8 1913.93  4876.1 1901.71  4900.6 1888.53  4907.1 1883.25
  4917.4 1879.35  4936.2 1868.45  4958.7 1860.89    4975  1858.9  4975.3  1858.4
    4979  1858.9  4982.2 1858.96  4997.4 1877.77    5003 1877.77  5007.6 1883.49
  5028.8 1889.27  5065.3 1910.43  5071.2  1910.8  5101.8 1921.03  5138.3 1928.22
  5211.3 1932.86  5372.9 1937.17    5393  1939.2  5405.5 1941.42  5478.5 1943.51
#Mann= 8 ,-1 , 0
  4536.1     .07       0    4604    .035       0  4729.9     .12       0
    4809     .07       0    4975     .05       0    4979     .07       0
  5372.9    .035       0    5393     .07       0
Bank Sta=4975,4979
XS Rating Curve= 0 ,0
Exp/Cntr=0.3,0.1

Type RM Length L Ch R = 1 ,68508   ,553,553,553
BEGIN DESCRIPTION:
BIG JOSHUA CREEK 128.0
END DESCRIPTION:
XS GIS Cut Line= 4
      1994944.92     13855129.67        1995475.       13855125.
      1995636.75      13855101.7      1996017.32     13854879.92
#Sta/Elev= 30
  4469.9 1953.55    4580 1947.36  4646.1 1941.07    4720 1937.29    4810 1929.74
    4860  1919.5    4890 1907.58    4920 1886.85    4970 1860.01  4997.5  1848.3
  5018.2 1841.72  5018.5 1841.22  5022.2 1841.72  5035.2 1842.24  5040.4 1844.35
  5050.5 1854.71  5060.6 1858.41  5121.2 1869.46  5157.6 1882.95    5167 1883.84
    5173 1888.58  5188.5 1893.46  5204.2 1903.02    5210 1903.93  5225.7 1911.27
  5284.4 1924.25  5392.9 1934.92  5444.9 1937.81  5482.1 1943.12  5603.9 1954.17
#Mann= 5 ,-1 , 0
  4469.9     .12       0  4646.1     .07       0  5018.2     .05       0
  5022.2     .07       0  5157.6     .12       0
Bank Sta=5018.2,5022.2
XS Rating Curve= 0 ,0
Exp/Cntr=0.3,0.1

Type RM Length L Ch R = 1 ,67955   ,737,737,737
BEGIN DESCRIPTION:
BIG JOSHUA CREEK 127.0
END DESCRIPTION:
XS GIS Cut Line= 3
      1995435.46     13855891.22        1995775.       13855525.
      1996089.05     13855140.18
#Sta/Elev= 30
  4500.6 1942.76  4598.3 1935.93  4695.8 1926.13  4768.4 1922.92    4816  1918.6
  4829.4 1915.19  4844.4 1909.97  4865.4 1895.23  4901.1 1878.67  4929.4 1861.29
  4936.2 1855.03  4986.1 1831.18  4994.6 1830.13  4994.8 1829.63  4998.6 1830.13
  5085.4 1843.17  5114.2 1849.52  5178.1 1874.69  5184.5 1880.35  5192.4 1882.58
  5198.9 1887.79  5213.2 1892.16  5234.1 1904.74    5242 1906.89  5262.8    1919
  5277.1 1924.79  5320.2 1930.87  5384.1 1935.82  5419.3 1941.95  5496.7 1947.92
#Mann= 6 ,-1 , 0
  4500.6     .07       0  4598.3    .035       0  4768.4     .07       0
  4829.4     .12       0  4994.6     .05       0  4998.6     .12       0
Bank Sta=4994.6,4998.6
XS Rating Curve= 0 ,0
Exp/Cntr=0.3,0.1

Type RM Length L Ch R = 1 ,67218   ,816,816,816
BEGIN DESCRIPTION:
BIG JOSHUA CREEK 126.0
END DESCRIPTION:
XS GIS Cut Line= 3
      1996047.32     13856268.56        1996275.       13856025.
       1996512.7     13855724.69
#Sta/Elev= 30
  4666.6 1920.85  4701.8 1917.91  4757.5 1916.56  4766.7  1916.7  4794.7 1913.29
  4822.9    1904  4851.3 1889.64  4901.1 1860.78  4950.4 1838.17  4957.7 1832.87
  4964.6 1825.95  4971.9 1822.16  4978.8 1812.88  4986.1 1806.18  4996.6 1802.45
  5005.2 1802.25  5005.5 1801.75  5009.2 1802.25    5028 1814.55  5056.9 1818.95
  5106.6 1843.04  5149.9 1859.79  5185.1 1877.07  5234.8 1895.48  5249.2 1902.54
    5270  1906.5  5278.1 1909.58  5292.5 1911.71  5348.6 1913.67    5383 1917.08
#Mann= 5 ,-1 , 0
  4666.6     .07       0  4701.8    .035       0  4757.5     .12       0
  5005.2     .05       0  5009.2     .12       0
Bank Sta=5005.2,5009.2
XS Rating Curve= 0 ,0
Exp/Cntr=0.3,0.1

Type RM Length L Ch R = 1 ,66402   ,753,753,753
BEGIN DESCRIPTION:
BIG JOSHUA CREEK 125.0
END DESCRIPTION:
XS GIS Cut Line= 3
      1996294.77     13856748.14        1996675.       13856675.
      1996925.69     13856381.88
#Sta/Elev= 30
  4612.8 1912.22  4694.5  1907.4  4771.5 1889.11  4786.2 1887.08  4837.1 1866.89
  4922.1 1826.94  4968.9 1800.57    4974 1801.47  4979.6  1795.4  4989.8 1790.62
  5011.7 1786.73    5012 1786.23  5015.7 1786.73    5050 1793.56  5056.5 1801.08
  5064.2 1800.42  5070.8 1814.18  5078.5 1819.25  5085.1 1827.95  5099.3 1831.27
  5120.2 1842.68  5127.9 1843.28  5134.5 1848.08  5170.7 1859.35  5177.3 1863.97
  5191.6 1866.57  5198.1 1870.75  5269.5 1895.51  5312.3  1906.3  5385.7  1910.7
#Mann= 4 ,-1 , 0
  4612.8    .035       0  4771.5     .12       0  5011.7     .05       0
  5015.7     .12       0
Bank Sta=5011.7,5015.7
XS Rating Curve= 0 ,0
Exp/Cntr=0.3,0.1

Type RM Length L Ch R = 1 ,65649   ,758,758,758
BEGIN DESCRIPTION:
BIG JOSHUA CREEK 124.0
END DESCRIPTION:
XS GIS Cut Line= 3
      1996402.23      13857117.9        1996725.       13857325.
      1997139.24     13857417.76
#Sta/Elev= 30
  4616.5 1884.18  4623.1  1881.8  4674.6  1875.7  4695.7 1870.04  4726.1 1866.84
  4747.3 1862.88  4753.2 1860.04  4841.1 1849.84  4869.3 1844.56  4898.6 1835.88
  4904.9 1830.35  4934.9 1811.88  4964.4 1796.46  4971.3 1788.29  4977.2 1787.09
  4986.5  1777.9  4990.4 1777.05  4990.7 1776.55  4994.4 1777.05  5024.3 1779.41
  5030.7 1785.98    5041 1790.02  5116.1 1808.24  5202.9 1843.25  5245.9 1856.73
  5251.4 1860.63  5266.4 1866.02  5317.7 1881.27  5384.3 1888.77  5424.5 1896.62
#Mann= 3 ,-1 , 0
  4616.5     .12       0  4990.4     .05       0  4994.4     .12       0
Bank Sta=4990.4,4994.4
XS Rating Curve= 0 ,0
Exp/Cntr=0.3,0.1

Type RM Length L Ch R = 1 ,64891   ,410,410,410
BEGIN DESCRIPTION:
BIG JOSHUA CREEK 123.0
END DESCRIPTION:
XS GIS Cut Line= 3
      1996032.22     13857564.37      1996324.96     13857887.48
      1996676.42     13857892.41
#Sta/Elev= 30
    4564 1880.33  4630.4 1863.42  4665.5 1848.29  4679.7 1847.92  4722.3 1834.09
    4729 1828.79  4750.7 1825.07  4757.4 1819.99  4764.9 1820.94  4771.6 1814.88
  4779.1  1815.5  4785.8 1808.69  4793.2 1810.12    4800  1804.2  4828.4 1800.68
  4849.3 1791.62  4906.1 1786.99  4920.3 1781.12  4941.9 1785.03  4956.1  1781.7
  4962.9 1771.77  4981.8 1765.99  4982.1 1765.49  4985.8 1765.99    5030 1774.02
    5060 1773.84  5090.1 1785.98  5120.1 1805.35  5200.1 1840.18  5351.5 1881.48
#Mann= 3 ,-1 , 0
    4564     .12       0  4981.8     .05       0  4985.8     .12       0
Bank Sta=4981.8,4985.8
XS Rating Curve= 0 ,0
Exp/Cntr=0.3,0.1

Type RM Length L Ch R = 1 ,64481   ,447,447,447
BEGIN DESCRIPTION:
BIG JOSHUA CREEK 122.0
END DESCRIPTION:
XS GIS Cut Line= 3
      1996374.99       13858275.        1996475.       13858225.
      1996725.03     13858174.99
#Sta/Elev= 30
  4883.5 1784.87  4928.2 1783.28  4936.6 1780.26  4950.6 1772.06    4959 1768.38
  4964.6 1766.96  4986.9 1766.47  4992.5 1764.99  4997.9 1764.99  5005.5 1763.39
  5013.1 1763.33  5013.5 1762.83  5018.3 1763.33  5036.1 1763.65  5046.3 1764.56
  5056.5 1767.21  5064.2 1770.62  5076.9 1777.54  5107.5 1790.18  5117.7 1796.11
  5122.8 1803.95  5127.9 1805.57  5138.1 1811.39  5158.5 1824.97  5168.7  1839.5
  5178.9 1852.25  5199.3 1865.08  5209.5 1870.08  5229.9 1876.39  5250.3 1878.66
#Mann= 4 ,-1 , 0
  4883.5     .07       0  5013.1     .05       0  5018.3     .07       0
  5064.2     .12       0
Bank Sta=5013.1,5018.3
XS Rating Curve= 0 ,0
Exp/Cntr=0.3,0.1

Type RM Length L Ch R = 1 ,64034   ,343,343,343
BEGIN DESCRIPTION:
BIG JOSHUA CREEK 121.0
END DESCRIPTION:
XS GIS Cut Line= 3
      1996174.99       13858925.        1996525.       13858625.
      1996725.01       13858525.
#Sta/Elev= 30
    4539  1887.5  4571.9 1883.31  4603.2 1875.64  4704.1 1838.32  4730.5 1822.43
  4751.4 1816.31  4759.1 1811.18    4837 1781.92  4879.8 1776.36    4950 1772.15
  4978.6 1764.13  4997.4 1767.92    5014 1767.47  5022.3  1763.8    5060 1763.79
  5072.8 1763.64  5073.3 1763.14  5078.1 1763.64  5103.4 1763.71  5111.8 1765.85
  5120.2 1772.28  5125.8 1772.59  5142.5 1788.42  5148.1  1788.1  5156.5 1801.12
  5164.9 1822.63  5170.5 1811.37  5178.9 1838.66  5201.2 1846.61  5223.6 1850.14
#Mann= 6 ,-1 , 0
    4539     .07       0  4704.1     .12       0  4997.4     .07       0
    5060     .12       0  5072.8     .05       0  5078.1     .12       0
Bank Sta=5072.8,5078.1
XS Rating Curve= 0 ,0
Exp/Cntr=0.3,0.1

Type RM Length L Ch R = 1 ,63691   ,93,93,93
BEGIN DESCRIPTION:
BIG JOSHUA CREEK 120.5
END DESCRIPTION:
XS GIS Cut Line= 4
      1996392.71     13859106.65       1996640.9      13858890.9
      1996710.45     13858817.75      1996851.03     13858663.49
#Sta/Elev= 30
  4670.8 1835.98  4675.6 1835.98  4680.7 1830.19  4687.3 1828.85  4751.9 1792.47
  4809.8 1769.71  4827.1 1769.04  4827.5 1768.54  4832.4 1769.04  4864.9 1770.28
  4893.4  1774.9  4936.1 1775.75  5035.2 1775.95  5112.9 1771.41  5127.1 1772.98
  5151.4 1780.81  5183.9 1792.61  5190.6 1793.33  5198.1 1797.83  5204.8 1798.21
  5212.2 1802.81    5219 1803.23  5233.2 1814.37    5240 1815.57  5247.4 1821.29
  5254.1 1821.92  5261.6 1827.35  5268.3 1828.46  5289.9 1839.15  5309.3 1843.71
#Mann= 5 ,-1 , 0
  4670.8     .12       0  4809.8     .07       0  4827.1     .05       0
  4832.4     .07       0  5151.4     .12       0
Bank Sta=4827.1,4832.4
XS Rating Curve= 0 ,0
Exp/Cntr=0.3,0.1

Type RM Length L Ch R = 1 ,63598   ,472,472,472
BEGIN DESCRIPTION:
BIG JOSHUA CREEK 120.0
END DESCRIPTION:
XS GIS Cut Line= 3
      1996407.48     13859189.08        1996675.       13858975.
      1996916.81     13858710.37
#Sta/Elev= 30
  4652.6  1848.5  4711.1 1823.23  4781.5 1787.41  4824.8 1770.09  4839.2 1768.32
  4888.8 1769.54  4895.2 1774.79  4903.2 1775.85  4944.8 1752.25  4964.6 1748.44
    4965 1747.94  4969.9 1748.44  5002.3 1757.51    5080 1758.52  5115.8 1768.21
  5144.2 1772.03  5200.3 1771.25  5254.6 1777.83  5264.4 1781.89  5271.2 1781.44
  5278.6 1786.55  5285.4 1786.35  5292.8 1792.28  5299.6 1792.38  5313.8 1804.72
  5320.5 1804.82  5327.9 1811.06  5334.7 1811.42  5342.1 1818.12  5353.7 1820.07
#Mann= 5 ,-1 , 0
  4652.6     .12       0  4839.2     .07       0  4964.6     .05       0
  4969.9     .07       0  5254.6     .12       0
Bank Sta=4964.6,4969.9
XS Rating Curve= 0 ,0
Exp/Cntr=0.3,0.1

Type RM Length L Ch R = 1 ,63126   ,466,466,466
BEGIN DESCRIPTION:
BIG JOSHUA CREEK 119.0
END DESCRIPTION:
XS GIS Cut Line= 3
        1997125.     13859425.01        1997075.       13859175.
      1997146.33     13858712.13
#Sta/Elev= 30
  4744.7  1844.9  4765.1 1841.05  4795.7 1828.29  4846.7 1803.33  4872.2  1793.9
  4877.3 1789.11  4938.5 1767.73  4969.1 1747.34  4979.3 1747.74  4986.8 1745.53
  4987.2 1745.03  4992.2 1745.53  5050.3    1751  5089.6 1751.51    5111 1750.58
  5121.1 1753.23  5141.3  1764.4  5151.4 1766.08  5181.8 1764.48  5303.2 1764.95
  5343.7 1767.37  5353.8 1769.79    5374 1778.41  5404.4 1794.69    5423 1807.98
  5428.1 1807.35  5434.7 1814.65    5455 1829.61    5464 1843.83    5468 1843.83
#Mann= 4 ,-1 , 0
  4744.7     .12       0  4986.8    .035       0  4992.2     .12       0
  5089.6     .12       0
Bank Sta=4986.8,4992.2
XS Rating Curve= 0 ,0
Exp/Cntr=0.3,0.1

Type RM Length L Ch R = 1 ,62660   ,500,500,500
BEGIN DESCRIPTION:
BIG JOSHUA CREEK 118.0
END DESCRIPTION:
XS GIS Cut Line= 3
      1997574.99     13859574.96        1997525.       13859225.
      1997874.99     13858825.01
#Sta/Elev= 30
  4646.5 1837.63  4727.7 1810.49  4757.6  1797.9    4798  1785.1  4818.2 1776.03
  4828.3 1765.73  4888.9 1758.25    4899 1751.39  4909.1 1750.02  4927.3 1743.71
  4969.7 1740.24  4977.1 1737.35  4977.5 1736.85  4982.6 1737.35  4997.5 1742.05
  5016.4 1743.14  5198.9 1752.06  5205.5 1750.78  5219.7  1752.1  5226.4 1749.97
  5248.2 1751.14  5269.1 1746.41  5276.7 1746.99  5283.3 1752.07  5332.7 1775.49
  5375.4 1800.34  5418.1 1827.93    5439 1844.73  5495.9 1863.91  5531.5 1871.44
#Mann= 6 ,-1 , 0
  4646.5     .07       0  4727.7     .12       0  4927.3    .035       0
  4977.1    .035       0  4982.6    .035       0  5016.4     .12       0
Bank Sta=4977.1,4982.6
XS Rating Curve= 0 ,0
Exp/Cntr=0.3,0.1

Type RM Length L Ch R = 1 ,62160   ,446,446,446
BEGIN DESCRIPTION:
BIG JOSHUA CREEK 117.0
END DESCRIPTION:
XS GIS Cut Line= 3
      1997624.99     13859625.01        1998025.       13859225.
      1998075.01     13859024.96
#Sta/Elev= 30
  4434.2 1842.61  4462.5 1841.64  4504.9  1826.4  4519.1 1820.45  4575.6 1789.21
  4610.4 1773.06  4632.2 1764.05  4660.5 1757.89  4688.8 1756.03  4800.4 1754.24
  4863.9 1753.68  4929.2 1751.48  4963.5 1748.93  4985.8 1735.04  4993.5  1733.6
    4994  1733.1  4999.2  1733.6  5023.1 1734.37  5041.1 1737.36  5051.4 1740.64
  5059.2 1746.08  5092.7 1760.58  5105.6 1768.32  5133.9 1788.47  5141.6 1796.22
  5146.8 1798.86  5154.5 1832.31  5164.8 1845.11  5182.9 1851.15  5206.1 1853.87
#Mann= 7 ,-1 , 0
  4434.2     .07       0  4610.4     .12       0  4800.4     .07       0
  4863.9    .035       0  4963.5     .12       0  4993.5     .05       0
  4999.2     .12       0
Bank Sta=4993.5,4999.2
XS Rating Curve= 0 ,0
Exp/Cntr=0.3,0.1

Type RM Length L Ch R = 1 ,61714   ,476,476,476
BEGIN DESCRIPTION:
BIG JOSHUA CREEK 116.0
END DESCRIPTION:
XS GIS Cut Line= 3
      1997701.87     13860283.37        1998375.       13859425.
      1998324.99     13859124.97
#Sta/Elev= 30
  3909.2 1883.59  3936.5 1881.69  4031.8 1878.51  4102.8 1871.49    4150  1869.1
    4272 1861.65  4365.4 1857.05    4394 1851.56  4458.5 1831.13  4522.7 1801.76
  4543.5 1791.08  4551.6 1781.23  4560.3 1779.58  4580.6 1777.44  4607.7 1762.58
  4651.1  1752.8    4799 1749.85  4878.9 1748.01  4959.6 1735.23  4975.4 1729.67
  4975.9 1729.17  4981.2 1729.67  5027.9 1731.99    5033 1729.94  5040.6 1732.39
  5060.9 1746.09  5093.8 1753.48  5154.6 1780.32  5253.5 1834.72  5304.2 1847.59
#Mann= 11 ,-1 , 0
  3909.2     .07       0  3936.5    .035       0  4102.8     .07       0
    4150    .035       0    4272     .07       0    4394     .12       0
  4560.3     .07       0    4799    .035       0  4959.6     .12       0
  4975.4     .05       0  4981.2     .12       0
Bank Sta=4975.4,4981.2
XS Rating Curve= 0 ,0
Exp/Cntr=0.3,0.1

Type RM Length L Ch R = 1 ,61238   ,466,466,466
BEGIN DESCRIPTION:
BIG JOSHUA CREEK 115.0
END DESCRIPTION:
XS GIS Cut Line= 3
      1998604.66      13860439.6        1998775.       13859625.
        1999175.       13859225.
#Sta/Elev= 30
  4167.8 1863.22  4212.2 1861.09  4245.9  1858.1  4290.8 1847.24  4390.7 1836.78
  4435.6 1822.83  4440.7 1826.83  4485.6  1809.1  4490.7 1812.95  4535.5  1795.5
  4540.6 1798.55  4594.5 1783.26  4630.4 1770.62  4635.5 1772.52  4694.4 1756.78
  4794.2 1748.21  4959.2 1742.45  4969.4 1740.93    4975 1733.82  4994.3 1724.54
  4994.8 1724.04  5000.6 1724.54  5135.6 1737.75  5162.9 1742.09  5325.3 1746.64
  5379.8 1756.32  5452.6 1782.54    5495 1806.83  5523.3 1829.92  5565.7 1848.01
#Mann= 10 ,-1 , 0
  4167.8     .07       0  4212.2     .12       0  4594.5     .07       0
  4694.4    .035       0  4794.2     .07       0  4994.3     .05       0
  5000.6     .07       0  5135.6    .035       0  5162.9     .07       0
  5379.8     .12       0
Bank Sta=4994.3,5000.6
XS Rating Curve= 0 ,0
Exp/Cntr=0.3,0.1

Type RM Length L Ch R = 1 ,60772   ,474,474,474
BEGIN DESCRIPTION:
BIG JOSHUA CREEK 114.0
END DESCRIPTION:
XS GIS Cut Line= 3
      1998824.97     13860075.03        1999225.       13859675.
      1999374.99     13859325.02
#Sta/Elev= 30
  4433.9    1817  4437.5    1817  4448.1 1812.27  4553.8 1775.68  4589.5  1763.2
  4635.9 1749.99  4674.4 1740.78  4697.7 1739.97  4773.4 1736.07  4886.5 1737.23
  4918.8 1734.94  4943.1 1732.09  4992.9 1719.67  4993.4 1719.17  4999.2 1719.67
  5014.1 1719.71  5043.2  1731.8  5061.3 1737.68  5130.2 1738.98    5161 1746.64
  5176.4 1753.81  5184.6 1756.65  5195.5 1762.59  5206.3 1765.61  5249.9  1786.8
  5260.7 1790.72  5336.9 1831.36  5347.8 1838.39  5365.9 1844.41  5380.4 1846.93
#Mann= 8 ,-1 , 0
  4433.9     .12       0  4553.8    .035       0  4635.9     .12       0
  4697.7    .035       0  4918.8     .07       0  4992.9     .05       0
  4999.2     .07       0  5176.4     .12       0
Bank Sta=4992.9,4999.2
XS Rating Curve= 0 ,0
Exp/Cntr=0.3,0.1

Type RM Length L Ch R = 1 ,60298   ,476,476,476
BEGIN DESCRIPTION:
BIG JOSHUA CREEK 113.0
END DESCRIPTION:
XS GIS Cut Line= 3
      1998975.02     13860374.98        1999325.       13860025.
      1999425.05       13860025.
#Sta/Elev= 30
  4505.6 1865.68  4509.1 1865.68  4533.9    1860  4562.1 1849.62  4576.3 1838.75
  4590.4 1821.02  4604.6  1808.9    4647 1781.58  4675.3 1766.02  4689.4 1759.41
  4731.9 1742.92    4746 1738.27  4774.3 1734.64  4824.3 1732.51  4842.7 1730.28
  4873.3 1725.15  4887.4 1725.51  4901.6 1723.69  4929.8 1722.38  5003.1 1720.26
  5010.6 1716.56  5017.4 1716.03  5017.9 1715.53  5023.7 1716.03  5030.6 1725.24
  5040.6 1731.13  5050.6 1733.64  5060.6 1734.75  5080.6 1735.85  5100.6  1735.6
#Mann= 5 ,-1 , 0
  4505.6     .07       0  4824.3    .035       0  4842.7     .07       0
  5017.4     .05       0  5023.7     .07       0
Bank Sta=5017.4,5023.7
XS Rating Curve= 0 ,0
Exp/Cntr=0.3,0.1

Type RM Length L Ch R = 1 ,59822   ,489,489,489
BEGIN DESCRIPTION:
BIG JOSHUA CREEK 112.0
END DESCRIPTION:
XS GIS Cut Line= 3
      1999225.03     13860524.98        1999325.       13860475.
      1999425.01     13860274.98
#Sta/Elev= 30
  4882.4  1854.9  4885.2  1854.9  4890.8 1850.22  4913.1 1836.86  4918.7  1805.8
  4927.1 1781.88  4935.5 1774.88  4941.1 1765.07  4949.4 1759.15  4957.8 1754.13
  4963.4 1747.38  4980.2 1738.82  4985.8 1731.87  4991.4 1718.86    4997 1718.86
  5002.6 1712.14  5004.9 1712.09  5005.4 1711.59  5011.3 1712.09  5024.9 1714.04
  5030.5 1717.53    5032 1717.67  5052.9 1719.07  5061.3 1720.48  5083.6 1720.65
    5106 1722.04  5119.9 1724.01  5164.7 1726.73    5187 1726.98  5217.8 1729.54
#Mann= 4 ,-1 , 0
  4882.4     .07       0  5004.9     .05       0  5011.3     .07       0
    5032    .035       0
Bank Sta=5004.9,5011.3
XS Rating Curve= 0 ,0
Exp/Cntr=0.3,0.1

Type RM Length L Ch R = 1 ,59333   ,469,469,469
BEGIN DESCRIPTION:
BIG JOSHUA CREEK 111.0
END DESCRIPTION:
XS GIS Cut Line= 4
      1999645.66     13860667.69      1999736.13     13860591.87
        1999775.       13860475.      1999780.51     13860188.16
#Sta/Elev= 30
  4754.1 1730.65  4783.7 1728.79  4792.5 1727.62  4798.1 1726.85  4818.9 1720.24
  4833.2 1717.75    4841 1717.61  4847.5 1716.75  4921.5 1715.96  4942.6 1714.42
  4947.8 1714.95  4963.7 1710.53  4974.2  1709.2  4997.8 1709.66  5005.3 1709.02
  5012.1 1707.15  5012.6 1706.65    5018 1706.65  5018.5 1707.15  5025.3 1709.36
  5035.3 1714.82  5045.3 1717.34  5055.3 1717.57  5075.3 1716.14  5115.3 1716.53
  5195.3 1722.72  5217.6 1723.62  5258.1 1723.89  5275.4 1726.85  5282.2 1726.53
#Mann= 6 ,-1 , 0
  4754.1     .12       0  4792.5    .035       0  5012.1    .035       0
  5018.5    .035       0  5115.3     .12       0  5217.6     .07       0
Bank Sta=5012.1,5018.5
XS Rating Curve= 0 ,0
Exp/Cntr=0.3,0.1

Type RM Length L Ch R = 1 ,58864   ,449,449,449
BEGIN DESCRIPTION:
BIG JOSHUA CREEK 110.0
END DESCRIPTION:
XS GIS Cut Line= 3
      2000021.63     13860718.85        2000175.       13860475.
      2000283.66     13860239.54
#Sta/Elev= 30
    4708 1728.21  4713.2 1728.21  4721.1 1732.58    4727 1733.41  4736.2 1732.78
  4742.3 1728.44  4757.6 1724.89  4802.3  1723.4  4836.5 1721.04    4873  1715.7
    4946 1713.39  4967.2 1709.13  4988.4 1709.39  4993.1 1706.07  5010.3 1702.91
  5012.3 1702.47  5012.8 1701.97    5024 1702.47  5056.2 1705.75  5073.2 1714.79
  5079.1 1721.92  5095.2 1725.14  5117.1 1726.37  5170.9 1729.37  5193.9 1728.43
  5199.4 1724.62  5238.4 1733.48  5245.3 1737.38  5250.8  1736.5  5255.4 1738.92
#Mann= 6 ,-1 , 0
    4708     .07       0  4802.3    .035       0  5010.3     .07       0
  5012.3    .035       0    5024     .07       0  5117.1     .12       0
Bank Sta=5012.3,5024
XS Rating Curve= 0 ,0
Exp/Cntr=0.3,0.1

Type RM Length L Ch R = 1 ,58415   ,471,471,471
BEGIN DESCRIPTION:
BIG JOSHUA CREEK 109.0
END DESCRIPTION:
XS GIS Cut Line= 3
      1999978.82      13861262.7        2000475.       13860725.
      2000624.97     13860625.02
#Sta/Elev= 30
  4263.7 1743.46  4408.2 1731.59  4450.7 1730.64  4506.8  1725.8  4633.4 1723.94
  4662.8 1725.35  4747.8 1718.99    4827 1718.07  4853.9 1716.36  4903.2 1709.43
  4945.7 1709.61  4964.2 1705.14  4998.4 1701.63  5002.9 1699.71  5025.5 1698.77
    5026 1698.27  5037.3 1698.77  5038.9 1701.99    5060 1712.27  5067.5 1741.59
    5081 1753.83    5090 1759.26  5099.4 1768.65    5111 1777.16    5117 1786.52
  5126.1 1792.03  5139.6 1806.24  5147.1 1841.17  5162.1 1847.84  5175.6 1849.24
#Mann= 7 ,-1 , 0
  4263.7    .035       0  4633.4     .07       0    4827    .035       0
  4964.2     .07       0  5025.5     .05       0  5037.3     .07       0
  5099.4     .12       0
Bank Sta=5025.5,5037.3
XS Rating Curve= 0 ,0
Exp/Cntr=0.3,0.1

Type RM Length L Ch R = 1 ,57944   ,421,421,421
BEGIN DESCRIPTION:
BIG JOSHUA CREEK 108.0
END DESCRIPTION:
XS GIS Cut Line= 3
      2000315.16     13861336.52        2000675.       13861125.
      2000894.01     13861001.16
#Sta/Elev= 30
  4583.1 1718.55  4752.5 1711.22  4851.9 1708.07  4912.6 1706.59  4919.3 1706.24
  4923.1 1704.82  4928.3 1702.88  4955.5 1701.72  4968.4 1699.33  5008.3  1697.1
  5008.8  1696.6  5020.1  1697.1  5029.2 1700.38  5057.9 1716.13  5083.9 1722.01
  5089.3 1723.64    5095 1722.84  5110.9 1729.24  5132.7 1729.57  5148.5 1733.28
  5170.1 1735.75  5175.9 1739.43  5184.3 1742.01  5191.8 1742.71  5197.5 1746.79
  5213.4 1748.92  5219.2 1753.64  5229.3 1754.92  5235.1 1759.66  5252.1 1760.92
#Mann= 8 ,-1 , 0
  4583.1     .07       0  4851.9    .035       0  4923.1     .07       0
  4968.4    .035       0  5008.3    .035       0  5020.1    .035       0
  5083.9     .07       0  5132.7     .12       0
Bank Sta=5008.3,5020.1
XS Rating Curve= 0 ,0
Exp/Cntr=0.3,0.1

Type RM Length L Ch R = 1 ,57523   ,450,450,450
BEGIN DESCRIPTION:
BIG JOSHUA CREEK 107.0
END DESCRIPTION:
XS GIS Cut Line= 3
      2000296.16     13861521.04        2000775.       13861475.
      2001121.74     13861436.67
#Sta/Elev= 30
  4523.5 1730.87  4535.9 1729.91  4572.6 1723.76  4582.6 1725.42  4602.7 1722.11
  4740.8 1710.12  4803.6 1705.82    4894 1704.75  4924.2 1697.15  4944.3 1697.56
  4988.5  1695.4    4989  1694.9  5000.5  1695.4    5002 1697.67  5034.7 1701.85
  5044.8 1706.16  5049.9 1709.53    5055 1703.94  5064.9 1705.81    5085 1712.86
  5115.2 1717.92  5125.3 1717.86  5145.8 1714.21  5155.5 1715.73  5165.5 1719.07
  5175.6 1719.65  5256.1 1720.83  5310.7  1720.1  5327.3 1721.21  5353.4 1719.83
#Mann= 4 ,-1 , 0
  4523.5    .035       0  4988.5     .05       0  5000.5    .035       0
  5310.7     .12       0
Bank Sta=4988.5,5000.5
XS Rating Curve= 0 ,0
Exp/Cntr=0.3,0.1

Type RM Length L Ch R = 1 ,57073   ,453,453,453
BEGIN DESCRIPTION:
BIG JOSHUA CREEK 106.0
END DESCRIPTION:
XS GIS Cut Line= 3
      2000625.01     13862174.99        2000775.       13861925.
      2001249.04      13861398.9
#Sta/Elev= 30
  4708.5 1828.38  4731.8 1823.37  4766.8 1795.56  4815.3 1762.98  4832.9  1748.1
  4848.4 1737.26  4854.3  1735.2  4860.1 1727.14  4869.8 1723.93  4875.6 1718.55
    4897 1708.06  4906.7  1705.6  4918.4 1697.38  4933.9 1692.42  4980.4 1690.36
  4980.9 1689.86  4992.5 1690.36  5035.5 1693.32  5069.3 1698.95  5106.5  1701.4
  5113.3 1704.14  5148.4 1708.41  5216.3 1709.84  5374.4 1712.02  5473.9 1714.25
  5526.9 1715.01  5602.7 1715.94  5651.4 1717.81  5679.4 1722.39  5708.2 1730.92
#Mann= 11 ,-1 , 0
  4708.5    .035       0  4815.3     .12       0  4980.4     .05       0
  4992.5     .12       0  5069.3    .035       0  5216.3     .07       0
  5374.4    .035       0  5473.9     .07       0  5526.9    .035       0
  5602.7     .07       0  5679.4     .12       0
Bank Sta=4980.4,4992.5
XS Rating Curve= 0 ,0
Exp/Cntr=0.3,0.1

Type RM Length L Ch R = 1 ,56620   ,466,466,466
BEGIN DESCRIPTION:
BIG JOSHUA CREEK 105.0
END DESCRIPTION:
XS GIS Cut Line= 3
      2001007.18     13862385.03        2001025.       13862225.
       2001281.8     13861400.06
#Sta/Elev= 30
  4839.4  1783.6  4859.5 1779.37  4864.7 1777.36  4869.8 1772.93  4879.7 1770.45
  4940.1 1759.12  4950.1 1757.74  4965.8 1749.67  4970.2 1747.93  4980.3 1734.76
  4997.9 1705.34    5003 1705.34  5010.9 1692.61  5015.9 1686.53  5016.4 1686.03
    5028 1686.53  5054.4  1689.7  5063.3 1692.34    5087 1694.68  5094.7 1698.07
  5136.6 1698.45  5168.7 1701.23  5199.4 1703.94  5270.7 1705.54  5602.3 1707.76
  5651.9 1709.81  5758.6 1712.16    5781 1714.06  5791.1 1713.84  5864.4 1736.65
#Mann= 10 ,-1 , 0
  4839.4    .035       0  4940.1     .07       0  4965.8    .035       0
  5015.9    .035       0    5028    .035       0  5168.7     .07       0
  5270.7    .035       0  5602.3     .07       0  5651.9    .035       0
    5781     .12       0
Bank Sta=5015.9,5028
XS Rating Curve= 0 ,0
Exp/Cntr=0.3,0.1

Type RM Length L Ch R = 1 ,56154   ,561,561,561
BEGIN DESCRIPTION:
BIG JOSHUA CREEK 104.0
END DESCRIPTION:
XS GIS Cut Line= 3
      2001133.33     13862569.14        2001475.       13862175.
       2001424.1     13861410.31
#Sta/Elev= 30
  4478.5 1748.87  4483.6 1748.87  4489.6 1744.98  4581.8 1719.54  4610.3 1717.72
  4631.1  1713.7  4730.9  1707.5  4921.7 1706.38  4950.2 1704.43  4957.9 1696.94
  4964.5 1697.42  4972.1  1686.9  4978.7 1687.03  4986.4 1682.87  4990.8  1682.7
  4991.3  1682.2  5002.9  1682.7  5030.2 1688.25  5070.3 1690.58  5075.3 1694.74
  5339.3 1701.86  5443.6 1702.84  5592.7 1705.13  5611.5 1705.89  5621.5  1708.4
  5671.6 1724.73  5677.2  1728.9  5682.2 1727.73  5761.6 1764.61  5766.5 1764.61
#Mann= 6 ,-1 , 0
  4478.5     .12       0  4990.8    .035       0  5002.9     .12       0
  5339.3     .07       0  5443.6    .035       0  5592.7     .12       0
#XS Ineff= 2 , 0
       0                  5045.1       0 1695.98
Permanent Ineff=
       F       F
Bank Sta=4990.8,5002.9
XS Rating Curve= 0 ,0
Exp/Cntr=0.3,0.1

Type RM Length L Ch R = 1 ,55593   ,370,370,370
BEGIN DESCRIPTION:
BIG JOSHUA CREEK 103.0
END DESCRIPTION:
XS GIS Cut Line= 4
      2001583.54     13862450.54      2001954.49     13862245.35
      2001988.34     13862030.97       2001977.8     13861674.48
#Sta/Elev= 30
    4353  1704.9  4476.4 1701.38  4676.3 1697.17  4742.1 1696.02  4908.9 1695.77
  4929.1 1693.68  4937.3 1690.94  4942.4  1690.9  4949.4 1687.71  4959.5 1685.27
  4983.3 1680.96  4983.8 1680.46  4995.5 1680.96  4999.9 1682.25  5030.4 1683.66
  5039.9 1687.71    5050 1690.81    5080 1691.68  5128.9 1695.07    5170 1697.63
    5190  1702.1    5200 1701.57  5227.5 1708.19    5270 1715.55  5275.6 1715.85
  5280.7 1713.09  5300.1 1715.27  5320.1 1719.41  5347.8 1727.89  5350.6 1727.89
#Mann= 7 ,-1 , 0
    4353     .12       0  4676.3    .035       0  4983.3    .035       0
  4995.5    .035       0  5030.4     .12       0  5128.9     .07       0
  5227.5     .12       0
#XS Ineff= 2 , 0
       0                  5046.6       0  1692.5
Permanent Ineff=
       F       F
Bank Sta=4983.3,4995.5
XS Rating Curve= 0 ,0
Exp/Cntr=0.3,0.1

Type RM Length L Ch R = 1 ,55223   ,443,443,443
BEGIN DESCRIPTION:
BIG JOSHUA CREEK 102.0
END DESCRIPTION:
XS GIS Cut Line= 4
      2001640.74     13862457.25      2002271.22     13862175.94
        2002275.       13862175.        2002475.       13862075.
#Sta/Elev= 30
  4309.6 1703.01  4545.2 1697.57  4670.6 1694.35  4820.8 1694.52  4911.4 1685.04
  4944.4 1681.72  4976.1 1677.58  4976.6 1677.08  4988.3 1677.58  4988.9 1679.94
  4994.3 1678.42  4999.3 1681.82  5006.7 1681.82  5012.3 1686.61  5020.9 1690.33
  5026.2    1694  5040.2 1697.25  5048.6 1704.16    5057  1713.7  5062.6 1714.27
  5079.4 1734.19  5093.3 1743.51  5129.7 1761.65  5146.4 1773.77  5152.2 1776.11
  5168.8 1790.97  5174.4 1793.99  5182.8 1823.24  5191.2 1856.09  5227.5 1863.83
#Mann= 8 ,-1 , 0
  4309.6     .12       0  4545.2    .035       0  4911.4     .07       0
  4944.4     .12       0  4976.1     .05       0  4988.3     .12       0
  5020.9     .07       0  5152.2     .12       0
Bank Sta=4976.1,4988.3
XS Rating Curve= 0 ,0
Exp/Cntr=0.3,0.1

Type RM Length L Ch R = 1 ,54780   ,451,451,451
BEGIN DESCRIPTION:
BIG JOSHUA CREEK 101.0
END DESCRIPTION:
XS GIS Cut Line= 3
      2002025.03       13862575.        2002225.       13862575.
      2002480.41     13862555.77
#Sta/Elev= 30
  4795.3 1694.04  4835.3 1691.61  4845.3 1689.78  4855.3 1687.02  4865.3 1684.99
  4875.3  1684.1  4915.3 1684.43  4949.2 1682.93  4975.3  1681.1  4985.3  1677.1
  4997.8 1676.61  5005.3 1674.79  5009.2 1674.55  5009.7 1674.05    5021 1674.05
  5021.5 1674.55    5048 1677.11  5061.2 1679.44  5066.2 1679.53  5085.5 1684.99
  5105.6 1683.28  5115.6 1686.04  5155.7 1690.42  5185.8    1698    5193 1700.44
    5198 1698.55  5215.9 1703.76  5225.9 1705.81  5235.9 1707.25  5251.4 1708.47
#Mann= 5 ,-1 , 0
  4795.3    .035       0  4949.2     .07       0  5009.2     .05       0
  5021.5     .07       0    5048     .12       0
Bank Sta=5009.2,5021.5
XS Rating Curve= 0 ,0
Exp/Cntr=0.3,0.1

Type RM Length L Ch R = 1 ,54329   ,466,466,466
BEGIN DESCRIPTION:
BIG JOSHUA CREEK 100.0
END DESCRIPTION:
XS GIS Cut Line= 3
      2001736.57     13863215.88        2002225.       13863025.
      2002625.01     13862624.99
#Sta/Elev= 30
  4475.7 1721.55  4545.3 1720.71  4575.1 1713.51  4659.3 1708.74  4683.8 1705.37
  4713.6 1704.84  4767.9 1699.19  4792.4 1694.39  4827.5 1692.36  4846.7 1688.54
  4876.6 1688.92  4906.4 1685.14  4930.9 1679.54  4978.6 1676.85  5007.9 1670.64
  5008.4 1670.14  5020.6 1670.64  5070.8 1674.41  5099.1 1682.33  5199.9 1684.17
  5323.7 1689.29  5343.8 1689.73    5389 1691.07  5396.1 1692.86  5424.4 1691.98
  5458.6 1696.13  5495.1 1703.94  5537.5 1721.29  5562.3 1734.77  5565.8 1734.77
#Mann= 8 ,-1 , 0
  4475.7    .035       0  4827.5     .12       0  5007.9     .05       0
  5020.6     .12       0  5199.9    .035       0  5323.7     .07       0
  5343.8    .035       0  5458.6     .12       0
Bank Sta=5007.9,5020.6
XS Rating Curve= 0 ,0
Exp/Cntr=0.3,0.1

Type RM Length L Ch R = 1 ,53863   ,488,488,488
BEGIN DESCRIPTION:
BIG JOSHUA CREEK 99.0
END DESCRIPTION:
XS GIS Cut Line= 3
        2002175.       13863525.        2002275.       13863475.
      2002679.44     13863109.55
#Sta/Elev= 30
  4888.3 1697.12  4924.6 1693.15    4933 1691.42  4941.4 1688.07    4947 1689.34
  4950.9 1685.66  4955.4 1681.41  4963.8 1671.59  4986.1 1667.96  5003.5 1668.44
  5007.2 1668.29  5007.6 1667.46  5008.1 1666.96  5019.8 1666.96  5020.3 1667.46
  5021.4 1669.96  5028.1 1670.26  5042.3 1672.69  5049.8 1675.06  5070.7 1676.17
  5078.2  1678.2  5084.9 1677.36  5092.4 1679.17  5170.1 1679.61  5237.7 1678.45
  5269.5 1677.68  5303.4 1678.39  5424.9 1684.13  5511.1 1687.16  5545.2 1688.53
#Mann= 6 ,-1 , 0
  4888.3     .07       0  4950.9     .12       0  5007.6     .05       0
  5020.3     .12       0  5237.7    .035       0  5511.1     .07       0
Bank Sta=5007.6,5020.3
XS Rating Curve= 0 ,0
Exp/Cntr=0.3,0.1

Type RM Length L Ch R = 1 ,53375   ,381,381,381
BEGIN DESCRIPTION:
BIG JOSHUA CREEK 98.0
END DESCRIPTION:
XS GIS Cut Line= 3
      2002565.51     13863903.08        2002625.       13863675.
      2002825.03     13863474.97
#Sta/Elev= 30
  4764.3 1684.36    4786 1683.35  4820.4 1682.15  4866.1 1678.53  4896.2  1677.5
  4901.4 1678.51  4932.1 1676.52  4948.3 1676.61  4958.7 1675.65    4969 1671.63
  4977.2 1666.33  4982.4 1667.68  4983.3  1663.2  4983.8  1662.7    4996  1663.2
  4997.4 1663.92  5017.6 1663.96  5070.7 1664.85    5099 1666.39  5106.1 1668.75
  5113.1 1667.95  5118.4 1668.62  5141.4 1672.14  5183.9 1674.42  5212.1 1673.81
  5226.3 1675.03  5240.4 1679.85  5253.3 1685.18  5268.7 1687.38  5282.9 1687.55
#Mann= 8 ,-1 , 0
  4764.3     .12       0    4786     .07       0  4932.1     .12       0
  4983.3     .05       0    4996     .12       0  5017.6    .035       0
  5118.4     .12       0  5253.3    .035       0
Bank Sta=4983.3,4996
XS Rating Curve= 0 ,0
Exp/Cntr=0.3,0.1

Type RM Length L Ch R = 1 ,52994   ,1029,1029,1029
BEGIN DESCRIPTION:
BIG JOSHUA CREEK 97.0
END DESCRIPTION:
XS GIS Cut Line= 3
      2002425.02     13864374.98      2002999.62     13863697.64
        2003025.     13863475.01
#Sta/Elev= 30
  4112.2 1784.96  4140.2 1774.32  4176.5 1764.62  4211.6 1750.29  4228.1 1739.69
  4246.7 1731.44  4268.7 1726.87  4294.3 1717.49  4324.7 1710.52  4374.4 1690.94
  4402.7 1689.33  4417.3 1690.43    4439 1686.29  4486.3 1683.05  4537.8 1678.57
  4566.4 1679.56  4708.1 1672.37  4871.8  1671.1  4921.2 1667.67    4942 1664.43
  4966.4 1663.85  4992.1 1659.85  4992.6 1659.35  5005.6 1659.85  5005.9 1661.33
  5013.2  1664.9  5030.1 1666.82    5098 1681.83  5179.8  1694.3  5224.5 1696.39
#Mann= 9 ,-1 , 0
  4112.2     .12       0  4294.3    .035       0  4417.3     .07       0
  4486.3    .035       0  4966.4     .07       0  4992.1     .05       0
  5005.6     .07       0  5030.1    .035       0    5098     .12       0
Bank Sta=4992.1,5005.6
XS Rating Curve= 0 ,0
Exp/Cntr=0.3,0.1

Type RM Length L Ch R = 1 ,51965   ,378,378,378
BEGIN DESCRIPTION:
BIG JOSHUA CREEK 96.0
END DESCRIPTION:
XS GIS Cut Line= 3
      2002625.04     13864874.98        2003225.       13864575.
      2003372.89     13863411.14
#Sta/Elev= 30
  4330.2 1804.61  4366.5  1792.2  4433.6 1763.81    4509 1735.72  4567.7 1720.97
  4636.8 1707.95  4665.6 1703.66  4746.6 1698.75  4799.7 1691.12  4897.6 1686.05
  4933.9 1679.42  4947.9 1665.55  4964.6 1662.01  4970.2  1658.2    4987 1655.65
  4991.3 1652.37  4991.8 1651.87    5005 1652.37  5043.5  1657.1  5083.4 1665.54
    5132 1669.41  5214.5 1668.44  5438.4 1666.45  5518.4 1669.32  5535.2 1671.92
  5938.5 1672.94  6092.9 1675.98  6153.2 1679.97    6170 1683.96  6174.2 1683.96
#Mann= 8 ,-1 , 0
  4330.2     .12       0  4636.8    .035       0  4991.3    .035       0
    5005    .035       0  5083.4     .07       0  5214.5    .035       0
  6092.9     .07       0    6170     .12       0
Bank Sta=4991.3,5005
XS Rating Curve= 0 ,0
Exp/Cntr=0.3,0.1

Type RM Length L Ch R = 1 ,51587   ,984,984,984
BEGIN DESCRIPTION:
BIG JOSHUA CREEK 95.0
END DESCRIPTION:
XS GIS Cut Line= 3
       2003524.8     13864843.49      2003555.18      13864448.5
      2003559.52     13863393.86
#Sta/Elev= 30
    4601 1680.74    4760 1678.22    4790    1674  4843.9 1674.69  4932.5 1673.92
  4990.6 1671.12  4996.4 1661.86  5001.4 1661.86  5010.7 1654.83  5020.7  1652.4
  5030.7 1652.77  5033.8 1650.91  5034.3 1650.41  5047.5 1650.91  5050.7 1652.98
  5070.7 1653.35  5110.7 1656.46  5120.7 1658.58  5139.1 1659.96  5170.7 1663.12
    5213 1663.13  5270.7  1662.3  5350.7 1663.47  5380.7 1667.68  5410.7 1669.01
  5430.7 1668.38  5820.7 1672.79  5930.7  1676.6    6003 1681.51  6051.8 1690.08
#Mann= 7 ,-1 , 0
    4601    .035       0  4843.9     .12       0  5033.8     .05       0
  5047.5     .12       0  5139.1     .07       0    5213    .035       0
    6003     .12       0
Bank Sta=5033.8,5047.5
XS Rating Curve= 0 ,0
Exp/Cntr=0.3,0.1

Type RM Length L Ch R = 1 ,50603   ,453,453,453
BEGIN DESCRIPTION:
BIG JOSHUA CREEK 94.0
END DESCRIPTION:
XS GIS Cut Line= 3
      2003711.26     13864916.34        2004225.       13864175.
      2004416.45     13864015.71
#Sta/Elev= 30
  4093.2 1678.62  4334.4 1674.66    4399 1667.67  4477.6  1664.8  4650.6 1665.22
  4710.1 1659.04  4764.4 1658.77  4813.6 1658.07    4931 1653.14  4980.8 1646.49
  4981.3 1645.99  4994.6 1646.49  5016.6 1649.91  5023.1 1673.87    5031  1689.4
  5037.5 1693.44  5080.4 1702.55  5100.4 1710.27  5123.4 1713.53  5129.9 1717.62
  5137.7 1716.33  5144.2 1720.75  5158.5  1718.2    5165 1722.86  5172.9 1720.64
  5193.7 1726.45  5201.5 1724.34  5222.3 1729.71  5236.6 1726.33  5244.2 1729.18
#Mann= 7 ,-1 , 0
  4093.2    .035       0  4710.1     .07       0  4764.4     .12       0
  4813.6     .07       0  4980.8     .05       0  4994.6     .07       0
  5100.4     .12       0
Bank Sta=4980.8,4994.6
XS Rating Curve= 0 ,0
Exp/Cntr=0.3,0.1

Type RM Length L Ch R = 1 ,50150   ,462,462,462
BEGIN DESCRIPTION:
BIG JOSHUA CREEK 93.0
END DESCRIPTION:
XS GIS Cut Line= 3
      2003828.62     13864995.37        2004375.       13864575.
        2004875.       13864225.
#Sta/Elev= 30
  4315.4 1676.33  4569.8  1671.5  4590.7 1667.36  4677.9 1662.28  4799.4 1660.75
    4848 1660.89    4883 1659.12  4918.7 1657.24  4941.4 1650.13  4990.6 1644.76
  4991.1 1644.26  5004.5 1644.76  5004.8 1646.02  5051.6 1648.89  5083.7 1654.13
  5184.8 1658.03  5245.9 1665.86  5271.1 1668.96  5285.5 1673.86  5321.7 1691.72
  5363.6 1714.69  5407.6 1741.71  5414.1  1747.3  5449.9 1769.35  5456.4 1775.72
  5485.6    1795  5500.4 1806.83    5551 1838.68  5578.5 1851.72  5615.1 1863.01
#Mann= 8 ,-1 , 0
  4315.4    .035       0  4677.9     .12       0  4799.4    .035       0
    4883     .12       0  4990.6     .05       0  5004.5     .12       0
  5051.6     .07       0  5245.9     .12       0
Bank Sta=4990.6,5004.5
XS Rating Curve= 0 ,0
Exp/Cntr=0.3,0.1

Type RM Length L Ch R = 1 ,49688   ,425,425,425
BEGIN DESCRIPTION:
BIG JOSHUA CREEK 92.0
END DESCRIPTION:
XS GIS Cut Line= 3
      2004167.14      13865147.3        2004575.       13864975.
      2005024.97     13864475.03
#Sta/Elev= 30
  4557.5  1673.7  4826.6 1669.24  4885.4 1664.64  4915.5 1658.94  4932.9 1652.43
  4978.5 1651.78  5000.4  1642.2  5000.9  1641.7  5014.3  1642.2  5047.8 1644.67
  5269.3 1656.82  5302.7 1662.25  5368.4 1676.23    5411 1687.95  5467.8 1713.45
  5496.2  1727.8  5531.3 1750.07  5559.7 1763.62  5566.4 1770.02  5573.9 1773.05
  5580.6 1779.74  5588.1 1783.54  5594.8 1790.81  5602.3 1794.29  5616.5 1806.97
  5623.2 1831.95  5630.7 1837.95  5637.4 1842.03  5644.9 1843.07  5672.9 1842.44
#Mann= 6 ,-1 , 0
  4557.5    .035       0  4915.5     .12       0  5000.4     .05       0
  5014.3     .12       0  5047.8     .07       0  5302.7     .12       0
Bank Sta=5000.4,5014.3
XS Rating Curve= 0 ,0
Exp/Cntr=0.3,0.1

Type RM Length L Ch R = 1 ,49263   ,467,467,467
BEGIN DESCRIPTION:
BIG JOSHUA CREEK 91.0
END DESCRIPTION:
XS GIS Cut Line= 3
      2004321.31     13865453.29        2004775.       13865325.
      2005161.17     13865207.93
#Sta/Elev= 30
  4524.3  1667.2  4578.9 1665.12  4647.1 1662.49  4694.4 1657.86  4725.6 1656.45
  4746.4 1653.34  4754.2 1651.37  4793.4  1648.8  4869.6 1647.35  4891.9 1646.15
  4905.7 1646.58    4923 1645.88  4939.6 1644.13  4964.6 1643.26  4985.4 1640.31
  4993.2 1637.38  4998.4 1637.38  4999.2 1636.36  4999.7 1635.86  5013.2 1636.36
  5017.5 1640.69  5027.1 1644.61  5044.2 1648.75  5149.1 1650.37  5180.7 1652.05
  5258.3 1657.32  5284.7 1660.05  5362.2 1665.87  5388.6    1670  5399.3 1671.97
#Mann= 9 ,-1 , 0
  4524.3    .035       0  4578.9     .12       0  4869.6    .035       0
  4999.2    .035       0  5013.2    .035       0  5044.2     .07       0
  5180.7    .035       0  5284.7     .07       0  5388.6     .12       0
Bank Sta=4999.2,5013.2
XS Rating Curve= 0 ,0
Exp/Cntr=0.3,0.1

Type RM Length L Ch R = 1 ,48796   ,479,479,479
BEGIN DESCRIPTION:
BIG JOSHUA CREEK 90.0
END DESCRIPTION:
XS GIS Cut Line= 3
      2004375.03     13866274.97        2004975.       13865725.
      2005351.06     13865637.97
#Sta/Elev= 30
    4191 1676.51  4247.4 1674.56  4261.6 1671.45  4312.5 1666.89  4339.9 1659.25
    4352 1657.73    4396 1654.09  4530.4  1651.8  4686.4 1645.04  4693.2 1646.58
  4799.9  1643.7  4920.1 1645.81  4941.1  1640.3  4962.7  1638.9  4969.4 1636.06
  4969.7 1634.45  4970.2 1633.95    4984 1634.45  4997.8  1634.8  5000.1 1637.04
  5023.7 1640.98  5074.4  1642.9  5148.6 1643.98    5178 1648.02  5189.7 1651.51
  5199.6 1656.85  5204.8 1656.39  5210.2 1662.45  5220.5 1663.45  5390.9 1667.23
#Mann= 8 ,-1 , 0
    4191    .035       0  4312.5     .07       0    4352    .035       0
  4969.7    .035       0    4984    .035       0  5000.1     .07       0
  5074.4    .035       0    5178     .07       0
Bank Sta=4969.7,4984
XS Rating Curve= 0 ,0
Exp/Cntr=0.3,0.1

Type RM Length L Ch R = 1 ,48317   ,466,466,466
BEGIN DESCRIPTION:
BIG JOSHUA CREEK 89.0
END DESCRIPTION:
XS GIS Cut Line= 3
      2004475.02     13866474.99        2005075.       13866175.
        2005225.       13865975.
#Sta/Elev= 30
  4329.2 1670.93  4387.9 1667.79  4471.7 1657.51  4516.5 1653.98  4538.8  1652.7
  4566.8 1652.56  4583.5 1650.58  4700.9 1644.11  4740.1 1641.07  4788.8 1640.46
  4835.1 1641.05  4902.2 1640.17  4932.9 1638.21  4941.3 1636.94  4946.9 1637.19
  4963.7 1634.84    5006 1632.69  5006.5 1632.19  5021.1 1632.69  5036.5 1633.34
  5042.7 1635.49  5057.3 1636.46  5063.5 1641.45  5078.1 1642.52  5086.5 1642.04
  5092.7 1644.28    5100 1645.28  5136.5 1646.53  5192.7 1650.88    5250 1652.91
#Mann= 4 ,-1 , 0
  4329.2    .035       0  4788.8     .07       0    5006     .05       0
  5021.1     .07       0
Bank Sta=5006,5021.1
XS Rating Curve= 0 ,0
Exp/Cntr=0.3,0.1

Type RM Length L Ch R = 1 ,47851   ,476,476,476
BEGIN DESCRIPTION:
BIG JOSHUA CREEK 88.0
END DESCRIPTION:
XS GIS Cut Line= 4
      2004749.75     13866711.24        2005125.       13866625.
      2005262.82     13866590.15      2005325.79      13866091.7
#Sta/Elev= 30
  4614.9 1651.81  4617.8 1649.96  4681.8 1645.74  4713.7 1644.72  4751.5 1644.76
  4756.6 1643.85  4799.4 1641.53  4856.3 1639.12  4917.8 1639.53  4933.1 1635.09
  4938.4 1629.96  4958.9 1630.14  4982.1 1628.59  4982.6 1628.09  4997.3 1628.59
  4997.4 1629.77  5002.5 1629.77  5017.9 1634.39  5056.2 1637.62  5177.5 1639.63
  5291.8 1638.35  5328.7 1635.42  5356.4 1637.38  5361.5 1636.78  5409.3 1637.93
  5441.7 1639.68  5449.7 1641.07  5469.8 1642.43  5500.3  1642.1  5644.5 1644.72
#Mann= 6 ,-1 , 0
  4614.9    .035       0  4982.1    .035       0  4997.3    .035       0
  5056.2     .07       0  5291.8    .035       0  5500.3     .07       0
Bank Sta=4982.1,4997.3
XS Rating Curve= 0 ,0
Exp/Cntr=0.3,0.1
