HEC-RAS study BIG JOSHUA CREEK.prj: BIG JOSHUA CREEK Base Level Engineering

--- BIG JOSHUA CREEK.g01 (geometry) --- (continued)

Type RM Length L Ch R = 1 ,47375   ,899,899,899
BEGIN DESCRIPTION:
BIG JOSHUA CREEK 87.0
END DESCRIPTION:
XS GIS Cut Line= 3
      2005475.01     13866975.02        2005425.       13866775.
      2005357.85      13866230.4
#Sta/Elev= 30
  4789.7 1654.82  4812.9  1653.5    4849 1648.96  4854.1 1648.98  4890.2 1644.18
  4895.4 1644.19  4903.1 1642.61  4944.3 1638.76    4965 1637.77  4972.7 1636.55
  4977.8 1632.38  4985.6 1629.66  4993.3 1625.79  4998.3 1624.99  4998.8 1624.49
  5013.2 1624.49  5013.7 1624.99  5026.1 1628.13    5039 1627.49  5056.3 1632.66
  5096.6 1637.57  5126.9 1637.37  5167.2 1638.61  5227.6 1637.23  5319.2  1636.8
  5378.8 1634.22    5409 1636.64  5459.4 1639.07  5499.7 1642.22  5544.6    1642
#Mann= 5 ,-1 , 0
  4789.7     .07       0  4944.3    .035       0  4998.3    .035       0
  5013.7    .035       0  5319.2    .035       0
Bank Sta=4998.3,5013.7
XS Rating Curve= 0 ,0
Exp/Cntr=0.3,0.1

Type RM Length L Ch R = 1 ,46476   ,451,451,451
BEGIN DESCRIPTION:
BIG JOSHUA CREEK 86.0
END DESCRIPTION:
XS GIS Cut Line= 3
        2005475.       13867075.        2006075.       13866625.
      2006674.98     13866275.01
#Sta/Elev= 30
  4240.9  1658.2  4333.6 1654.13  4390.9 1643.94  4404.4  1644.1  4490.9 1636.16
  4662.8 1630.79  4883.6  1629.6  4940.9 1625.12  4948.2 1622.98  4977.4 1622.23
  4983.6 1623.86  4987.8 1620.61  4990.9 1620.61    4991 1618.84  4991.5 1618.34
  5006.5 1618.84  5048.8 1618.99  5063.3 1622.66  5071.9 1633.64    5079 1635.65
  5137.7 1635.17  5319.6 1643.13  5407.7 1643.71  5467.6 1646.52  5488.7 1647.87
  5501.5 1651.46  5523.4 1650.89  5597.5 1659.73  5656.2 1669.37  5685.5 1676.81
#Mann= 4 ,-1 , 0
  4240.9    .035       0    4991    .035       0  5006.5    .035       0
  5467.6     .07       0
Bank Sta=4991,5006.5
XS Rating Curve= 0 ,0
Exp/Cntr=0.3,0.1

Type RM Length L Ch R = 1 ,46025   ,638,638,638
BEGIN DESCRIPTION:
BIG JOSHUA CREEK 85.0
END DESCRIPTION:
XS GIS Cut Line= 3
      2005924.99     13867175.01        2006075.       13867025.
      2006675.02     13866424.98
#Sta/Elev= 30
  4783.6 1639.55  4858.3 1638.85  4910.9 1634.17    4925 1633.57  4939.2 1633.29
  4967.5 1634.46  4972.8 1628.15  4984.5 1614.41    4985 1613.91  4999.5 1613.91
    5000 1614.41  5031.1 1617.03  5038.2 1618.38  5108.9 1626.89  5202.3 1628.35
  5250.3 1627.78  5363.4 1629.76  5504.9 1634.59  5547.3 1636.51  5589.7 1637.31
  5632.1 1641.02  5660.4  1642.8  5674.6 1644.58  5688.7 1642.89  5715.4 1649.35
  5745.3  1653.2  5759.4  1655.8  5773.6 1656.38  5840.7 1666.07  5844.3 1666.07
#Mann= 7 ,-1 , 0
  4783.6    .035       0  4858.3    .045       0  4972.8     .07       0
  4984.5     .05       0    5000     .07       0  5202.3    .035       0
  5715.4     .07       0
Bank Sta=4984.5,5000
XS Rating Curve= 0 ,0
Exp/Cntr=0.3,0.1

Type RM Length L Ch R = 1 ,45387   ,400,400,400
BEGIN DESCRIPTION:
BIG JOSHUA CREEK 84.0
END DESCRIPTION:
XS GIS Cut Line= 3
      2006101.54     13867427.49      2006625.96      13866973.9
      2006851.72     13866369.56
#Sta/Elev= 30
  4308.3 1636.59  4516.6 1629.63  4631.6 1628.35  4823.1 1626.52  4851.6 1623.34
  4858.2 1619.45  4865.8 1621.12  4872.4 1616.23  4880.1 1617.83  4886.7 1613.79
  4915.2 1614.49  4989.9 1608.86  4990.4 1608.36  5005.6 1608.86  5021.8 1609.38
  5034.5 1614.81  5085.9 1621.84  5216.3  1626.6  5241.2 1638.09  5271.5 1641.86
  5326.8 1659.39  5357.1 1662.71  5382.1  1671.4  5528.2 1702.23  5553.2  1705.3
  5558.5  1709.3  5583.5 1713.55  5588.8 1718.33  5638.8 1726.17  5646.8 1731.08
#Mann= 6 ,-1 , 0
  4308.3    .035       0  4516.6    .045       0  4631.6    .035       0
  4989.9    .035       0  5005.6    .035       0  5034.5     .07       0
Bank Sta=4989.9,5005.6
XS Rating Curve= 0 ,0
Exp/Cntr=0.3,0.1

Type RM Length L Ch R = 1 ,44987   ,299,299,299
BEGIN DESCRIPTION:
BIG JOSHUA CREEK 83.0
END DESCRIPTION:
XS GIS Cut Line= 3
      2006324.98     13867475.02      2006985.09     13866984.85
      2007475.54     13866463.06
#Sta/Elev= 30
  4177.8 1634.36  4335.4 1629.12  4506.4 1619.92  4560.2 1619.96  4590.7 1620.21
  4813.1 1622.08  4907.5 1619.25  4986.3 1610.21  5005.9 1604.52  5006.4 1604.02
  5021.6 1604.52  5035.2 1623.03  5042.1 1626.21  5140.5 1627.97  5233.1 1636.94
  5282.9 1648.41  5303.9 1649.08  5346.4 1664.37  5410.8 1699.59  5544.6 1781.04
  5615.5 1817.92  5622.3 1818.53  5629.6 1823.25  5636.5 1822.35  5643.8 1826.87
  5650.6 1826.05  5657.9 1830.02    5679 1831.76  5693.1 1835.84  5716.1 1836.95
#Mann= 8 ,-1 , 0
  4177.8    .035       0  4560.2     .07       0  4590.7    .035       0
  4907.5     .07       0  5005.9     .05       0  5021.6     .07       0
  5140.5    .035       0  5410.8     .12       0
Bank Sta=5005.9,5021.6
XS Rating Curve= 0 ,0
Exp/Cntr=0.3,0.1

Type RM Length L Ch R = 1 ,44688   ,966,966,966
BEGIN DESCRIPTION:
BIG JOSHUA CREEK 82.0
END DESCRIPTION:
XS GIS Cut Line= 4
      2006480.85     13867423.99      2006804.07     13867259.07
      2007016.87     13867231.07      2007291.55     13867227.55
#Sta/Elev= 30
  4422.5 1629.27  4460.8 1626.42  4512.4 1623.52  4576.7 1620.73  4624.8 1617.89
  4737.3 1619.07  4765.4 1619.61  4816.6 1618.47  4853.4  1613.2  4858.4 1614.49
  4887.2 1613.12  4917.4 1613.39    4927 1611.99  4932.1 1614.17  4937.6 1613.26
  4947.7 1610.21  4957.8  1608.4    5000 1604.74  5000.3 1603.69  5000.8 1603.19
  5015.5 1603.19    5016 1603.69  5028.1 1606.37  5038.1 1623.27  5048.1 1625.46
  5058.1 1624.37  5083.4 1623.46  5088.4 1623.79  5188.1 1622.97  5274.7 1623.98
#Mann= 7 ,-1 , 0
  4422.5    .035       0  4512.4     .07       0  4576.7    .035       0
  4624.8     .07       0  4737.3    .035       0  5000.3    .035       0
    5016    .035       0
Bank Sta=5000.3,5016
XS Rating Curve= 0 ,0
Exp/Cntr=0.3,0.1

Type RM Length L Ch R = 1 ,43722   ,457,457,457
BEGIN DESCRIPTION:
BIG JOSHUA CREEK 81.0
END DESCRIPTION:
XS GIS Cut Line= 3
      2006623.78     13867968.46        2007025.       13867775.
       2007253.1     13867274.01
#Sta/Elev= 30
  4548.4 1633.54  4688.1  1630.3  4702.8 1628.47  4789.2    1624  4866.7 1618.72
  4872.2 1615.26  4882.8 1613.92  4894.8 1609.21  4911.9 1610.41  4917.5 1607.18
  4949.4 1605.29  4957.1 1607.41  4962.7  1601.2  4971.6 1596.83  4979.7 1602.73
  4985.3 1597.47    5000 1596.54  5000.5 1596.04  5016.2 1596.54  5032.8 1597.28
  5048.7 1599.52  5054.2 1598.83  5059.8  1605.2  5070.7 1609.92  5077.3  1614.8
  5092.7 1615.38  5128.9 1613.48  5194.7  1614.4  5445.1 1622.78  5544.3 1622.54
#Mann= 7 ,-1 , 0
  4548.4    .035       0  4688.1     .07       0  4789.2    .035       0
    5000    .035       0  5016.2    .035       0  5032.8     .07       0
  5194.7    .035       0
Bank Sta=5000,5016.2
XS Rating Curve= 0 ,0
Exp/Cntr=0.3,0.1

Type RM Length L Ch R = 1 ,43265   ,452,452,452
BEGIN DESCRIPTION:
BIG JOSHUA CREEK 80.0
END DESCRIPTION:
XS GIS Cut Line= 4
      2007275.18     13868206.57      2007390.95     13867997.08
        2007425.       13867775.      2007476.44     13867501.42
#Sta/Elev= 30
  4536.3 1621.13    4545 1620.75  4572.5 1616.89  4582.9 1616.68  4588.6  1615.7
  4632.1 1613.58  4648.1 1613.51  4653.9 1612.86  4729.5 1612.12  4775.7 1610.23
  4858.7 1610.06  4878.9 1610.92    4889 1609.98  4909.3 1605.07  4929.5 1601.96
  4939.6 1599.93  4949.7 1596.72    4982 1595.74  4982.5 1595.24    4998 1595.24
  4998.5 1595.74  5020.7 1595.94  5026.6 1605.99  5042.2 1608.63  5051.2 1608.47
    5074 1609.79  5136.7 1612.13  5189.2 1616.37  5246.7 1619.67  5278.7  1622.4
#Mann= 5 ,-1 , 0
  4536.3    .035       0    4982    .035       0  4998.5    .035       0
  5042.2     .07       0    5074    .035       0
Bank Sta=4982,4998.5
XS Rating Curve= 0 ,0
Exp/Cntr=0.3,0.1

Type RM Length L Ch R = 1 ,42813   ,620,620,620
BEGIN DESCRIPTION:
BIG JOSHUA CREEK 79.0
END DESCRIPTION:
XS GIS Cut Line= 3
      2006810.41      13868684.6        2007775.       13868025.
      2008275.02     13867424.98
#Sta/Elev= 30
  3831.2 1644.41    4137 1631.43  4250.8 1629.43  4272.9  1625.5  4322.5 1623.96
  4409.9 1615.38  4444.2 1611.18    4481 1613.45  4546.7 1605.19  4648.3 1604.03
  4869.7  1607.6  4899.5 1601.42  4963.4 1598.06  4986.2 1592.47  5019.4 1591.07
  5019.9 1590.57    5036 1591.07    5042 1594.91  5064.2 1596.45    5085 1601.78
  5091.5 1608.21  5290.7 1621.54  5397.4 1640.99  5541.3 1662.35  5574.4 1667.11
    5646  1683.7  5695.5 1691.27  5730.7 1704.83  5752.8 1716.96  5780.8    1722
#Mann= 7 ,-1 , 0
  3831.2    .035       0  4409.9     .07       0  4444.2    .035       0
  5019.4    .035       0    5036    .035       0  5541.3    .035       0
    5646     .07       0
Bank Sta=5019.4,5036
XS Rating Curve= 0 ,0
Exp/Cntr=0.3,0.1

Type RM Length L Ch R = 1 ,42193   ,268,268,268
BEGIN DESCRIPTION:
BIG JOSHUA CREEK 78.0
END DESCRIPTION:
XS GIS Cut Line= 5
      2006866.82     13868719.33      2007313.86     13868367.77
      2007600.32      13868445.9      2007756.57     13868415.52
      2008034.33     13867990.19
#Sta/Elev= 30
  4253.7 1643.84  4462.1  1634.1  4611.2  1629.5  4683.5 1624.49  4733.2 1619.01
  4797.4 1617.36  4803.7 1615.08  4815.5 1616.16  4818.2 1616.48  4820.6 1613.13
  4829.8 1613.27    4835 1615.93  4854.7 1611.35  4869.6    1607  4885.8 1597.72
  4904.1 1593.71  4943.8 1593.52  5001.9  1587.4  5002.4  1586.9  5018.5  1587.4
  5051.6 1588.09  5057.9 1598.22    5063  1603.8  5124.3 1605.58    5155 1609.18
  5200.2 1609.94  5384.5 1611.43  5632.2 1610.05  5635.2 1609.95  5786.5 1610.46
#Mann= 8 ,-1 , 0
  4253.7    .035       0  4815.5     .07       0  5001.9     .05       0
  5018.5     .07       0  5200.2    .035       0  5384.5     .07       0
  5632.2    .035       0  5635.2     .07       0
Bank Sta=5001.9,5018.5
XS Rating Curve= 0 ,0
Exp/Cntr=0.3,0.1

Type RM Length L Ch R = 1 ,41925   ,454,454,454
BEGIN DESCRIPTION:
BIG JOSHUA CREEK 77.0
END DESCRIPTION:
XS GIS Cut Line= 4
      2007104.76     13868591.85        2007275.       13868575.
      2007786.95      13868467.6      2008047.35     13868020.58
#Sta/Elev= 30
    4824 1629.72  4874.5 1626.43  4942.1 1611.42  4947.1 1617.01  4954.9 1615.56
    4985 1604.88  4992.6 1596.09  4997.6 1596.09  5005.3 1592.76  5017.4  1584.2
  5017.9  1583.7    5034  1584.2  5035.9 1585.67  5056.4 1587.64  5107.9  1589.8
  5138.1 1590.61  5164.6 1596.14  5169.7 1595.41  5199.4  1598.1  5209.4  1600.5
  5214.5 1599.38  5219.9 1601.24  5251.6 1603.71  5291.4 1603.01    5394 1607.06
  5414.1 1608.43  5655.4 1611.11  5743.2 1610.28  5953.5 1609.68  6035.5 1609.45
#Mann= 9 ,-1 , 0
    4824    .035       0  5017.4    .035       0    5034    .035       0
  5107.9    .035       0  5251.6     .07       0    5394    .035       0
  5655.4     .07       0  5743.2    .035       0  5953.5     .07       0
Bank Sta=5017.4,5034
XS Rating Curve= 0 ,0
Exp/Cntr=0.3,0.1

Type RM Length L Ch R = 1 ,41471   ,440,440,440
BEGIN DESCRIPTION:
BIG JOSHUA CREEK 76.0
END DESCRIPTION:
XS GIS Cut Line= 4
        2007175.       13869125.        2007325.       13868975.
      2007656.74      13868801.8       2008073.4     13868016.23
#Sta/Elev= 30
  4792.9 1647.09  4835.3 1642.23  4849.5 1637.62  4863.6 1634.96  4891.9  1633.1
    4906 1629.11  4920.2 1622.39  4934.3 1608.67  4944.4 1601.55  4948.5 1598.66
  4962.6 1593.71  4969.7 1583.51  4982.5 1582.69    4983 1582.19  4999.2 1582.69
  5035.3 1586.31    5041 1588.22  5079.5 1593.03  5117.8 1594.93  5162.2 1594.79
  5196.8 1599.07  5316.8 1597.61  5348.7 1598.85  5379.3 1599.06  5466.1  1603.6
  5537.7 1602.62  5658.3 1607.41  5834.2 1610.25  6202.6 1609.23  6268.5 1609.43
#Mann= 6 ,-1 , 0
  4792.9    .035       0  4944.4     .07       0  4982.5     .05       0
  4999.2     .07       0  5348.7    .035       0  6202.6     .07       0
Bank Sta=4982.5,4999.2
XS Rating Curve= 0 ,0
Exp/Cntr=0.3,0.1

Type RM Length L Ch R = 1 ,41031   ,390,390,390
BEGIN DESCRIPTION:
BIG JOSHUA CREEK 75.0
END DESCRIPTION:
XS GIS Cut Line= 3
        2007575.     13869425.02        2007625.       13869225.
      2008099.46     13868024.86
#Sta/Elev= 30
    4794 1640.45  4812.1 1640.81  4817.2 1639.72  4853.3 1638.36  4886.8 1625.15
  4894.5 1620.78  4917.7  1615.9  4935.7  1610.1  4940.1 1610.74  4958.9 1608.77
  4969.2 1597.66    4977 1582.51  4981.5 1580.55    4982 1580.05  4998.2 1580.55
    5015 1582.29  5032.4 1582.11  5039.4  1584.3  5080.3 1586.79  5123.2 1590.35
  5236.7 1590.11  5277.8 1594.59  5423.3 1595.71  5494.8 1601.75  5561.2 1600.15
  5656.1 1605.91  5849.7 1609.01  6260.3 1609.17  6272.6 1609.19  6290.7 1609.26
#Mann= 8 ,-1 , 0
    4794    .035       0  4940.1     .12       0  4981.5     .05       0
  4998.2     .12       0  5080.3     .07       0  5277.8    .035       0
  6260.3     .07       0  6272.6    .035       0
Bank Sta=4981.5,4998.2
XS Rating Curve= 0 ,0
Exp/Cntr=0.3,0.1

Type RM Length L Ch R = 1 ,40641   ,499,499,499
BEGIN DESCRIPTION:
BIG JOSHUA CREEK 74.0
END DESCRIPTION:
XS GIS Cut Line= 3
      2008175.02     13869175.01      2007956.22      13869070.9
      2008125.49     13868042.24
#Sta/Elev= 30
  4764.5 1617.21  4795.8  1616.6  4821.1 1607.87    4831 1603.32  4846.8 1599.68
  4875.3 1596.39  4920.5 1595.24  4965.9  1596.1  4974.9  1594.2    4983 1586.66
  4988.6 1579.93  5014.5 1577.48    5015 1576.98  5031.3 1577.48    5047 1578.24
  5053.3  1578.2  5090.2 1585.01  5095.3 1584.04  5151.4 1586.73  5225.6 1587.67
    5256  1595.9  5278.9  1596.7  5306.7 1595.88  5428.3 1598.52  5457.4 1600.36
  5462.5  1599.8  5539.8 1605.57  5584.9 1605.18  5732.3  1608.2  6049.3 1608.97
#Mann= 5 ,-1 , 0
  4764.5    .035       0  4821.1     .07       0  5014.5     .05       0
  5031.3     .07       0    5047    .035       0
Bank Sta=5014.5,5031.3
XS Rating Curve= 0 ,0
Exp/Cntr=0.3,0.1

Type RM Length L Ch R = 1 ,40142   ,446,446,446
BEGIN DESCRIPTION:
BIG JOSHUA CREEK 73.0
END DESCRIPTION:
XS GIS Cut Line= 3
      2008375.01     13868975.04        2008325.       13868775.
      2008338.17     13868185.45
#Sta/Elev= 30
  4793.5 1612.36  4834.8 1613.21  4845.1    1611  4852.8 1607.41    4858 1602.92
  4865.7 1598.85    4876 1594.85  4917.2 1582.22  4935.3 1579.59  4940.4 1579.57
  4948.2 1577.84  4968.8 1577.13    4981 1575.32  4981.5 1574.82  4997.8 1575.32
  4999.7 1576.85  5019.7 1576.97  5029.7 1581.73  5039.7 1587.64  5049.7 1590.87
  5079.7 1591.48  5152.6 1590.64  5219.2 1591.75  5224.2 1591.15  5351.5 1596.26
  5399.8 1599.28  5449.8  1604.3  5499.8 1604.11  5552.6 1606.51  5589.4  1605.8
#Mann= 6 ,-1 , 0
  4793.5     .07       0    4981     .05       0  4997.8     .07       0
  5152.6    .035       0  5351.5     .07       0  5552.6    .035       0
Bank Sta=4981,4997.8
XS Rating Curve= 0 ,0
Exp/Cntr=0.3,0.1

Type RM Length L Ch R = 1 ,39696   ,463,463,463
BEGIN DESCRIPTION:
BIG JOSHUA CREEK 72.0
END DESCRIPTION:
XS GIS Cut Line= 3
        2008675.     13868724.97        2008675.       13868525.
        2008625.     13868225.01
#Sta/Elev= 30
  4825.6 1609.35  4835.6 1608.65  4855.6 1609.52  4895.6  1609.4  4905.6 1607.72
  4915.6 1597.72  4925.6 1591.87  4955.6 1578.99  4965.6 1576.06  4997.2 1573.02
  4997.7 1572.52  5013.5 1572.52    5014 1573.02  5015.6 1573.49  5045.8 1574.11
  5053.4 1576.28  5058.5 1576.78  5076.3 1576.63  5085.9 1577.55  5096.5  1580.4
  5106.7 1581.77  5147.2  1583.1  5180.2 1586.11  5228.3 1589.37    5241 1591.93
  5258.7 1598.18  5265.1 1599.67    5279 1602.47  5296.8 1604.53  5329.7 1603.93
#Mann= 5 ,-1 , 0
  4825.6     .07       0  4997.2     .05       0    5014     .07       0
  5085.9    .035       0  5265.1     .07       0
Bank Sta=4997.2,5014
XS Rating Curve= 0 ,0
Exp/Cntr=0.3,0.1

Type RM Length L Ch R = 1 ,39233   ,448,448,448
BEGIN DESCRIPTION:
BIG JOSHUA CREEK 71.0
END DESCRIPTION:
XS GIS Cut Line= 3
      2008750.86     13869013.07        2008975.       13868225.
      2008885.11     13867669.45
#Sta/Elev= 30
  4185.9 1608.02  4214.6 1603.75  4290.5 1599.51  4306.2 1594.19  4350.2 1587.89
  4399.6 1589.91  4508.9 1589.05  4695.4 1587.04  4755.7 1587.74  4810.4  1584.7
  4818.1 1582.18  4876.3 1577.02  4881.5 1579.11  4901.3 1572.76  4931.1 1571.12
  4954.4 1570.67  4963.6 1567.06  4986.4 1565.66  4986.9 1565.16  5003.3 1565.66
  5015.7 1565.98  5025.5 1573.73  5055.9 1587.48  5086.3 1589.64  5100.3 1594.08
  5184.3 1599.87  5311.5 1607.13  5461.1  1616.9  5552.3 1630.33    5568 1633.06
#Mann= 13 ,-1 , 0
  4185.9    .035       0  4290.5     .07       0  4306.2    .035       0
  4508.9     .07       0  4695.4    .035       0  4810.4     .07       0
  4931.1    .063       0  4986.4     .05       0  5003.3    .063       0
  5015.7     .07       0  5184.3    .035       0  5311.5     .07       0
  5552.3     .12       0
Bank Sta=4986.4,5003.3
XS Rating Curve= 0 ,0
Exp/Cntr=0.3,0.1

Type RM Length L Ch R = 1 ,38785   ,464,464,464
BEGIN DESCRIPTION:
BIG JOSHUA CREEK 70.0
END DESCRIPTION:
XS GIS Cut Line= 3
      2008479.99     13869479.86        2009375.       13868275.
      2009293.03     13867703.76
#Sta/Elev= 30
  3503.4 1623.06  3625.2 1614.62  3765.4 1609.42  3824.1 1606.97  3889.3 1604.43
  3996.6 1606.31  4068.7 1606.11  4074.9 1601.76  4089.5 1604.87  4095.8 1600.47
  4139.6 1592.97  4160.4 1582.31  4175.1 1580.27  4393.1 1580.38  4783.8 1585.15
    4826 1583.47  4967.7 1558.96  4968.2 1558.46  4984.6 1558.96  5006.8 1565.12
  5014.4 1581.64  5024.5 1590.57  5034.5 1593.03  5039.6 1589.34  5052.8  1594.2
  5392.4 1606.54    5469 1615.62  5519.5 1629.75    5552 1634.98  5581.4 1640.87
#Mann= 11 ,-1 , 0
  3503.4     .07       0  3625.2    .035       0  3765.4     .07       0
  3824.1    .035       0  3996.6     .07       0  4393.1    .035       0
  4783.8     .07       0  4967.7     .05       0  4984.6     .07       0
  5052.8    .035       0    5552     .12       0
Bank Sta=4967.7,4984.6
XS Rating Curve= 0 ,0
Exp/Cntr=0.3,0.1

Type RM Length L Ch R = 1 ,38321   ,468,468,468
BEGIN DESCRIPTION:
BIG JOSHUA CREEK 69.0
END DESCRIPTION:
XS GIS Cut Line= 3
      2009325.01     13868824.99        2009475.       13868675.
      2009674.98     13868575.01
#Sta/Elev= 30
  4778.4 1592.77  4820.8 1593.19  4855.9 1592.39  4891.5 1592.13  4933.9 1593.68
  4948.1 1591.59  4962.2 1570.51  4976.4 1563.62    4987 1559.97  4993.3 1559.97
  4998.9 1558.92  5012.9 1559.23  5017.4  1558.5  5017.9    1558  5035.9    1558
  5036.4  1558.5  5057.6 1558.78    5080 1560.97  5088.3 1563.43  5102.3 1564.73
  5116.3  1567.6  5124.7 1567.06  5133.1 1571.42  5138.7 1576.01  5155.4 1585.47
    5161 1587.13  5169.4 1588.62  5183.4 1589.59  5191.8  1591.2  5214.1 1593.57
#Mann= 4 ,-1 , 0
  4778.4    .035       0  4855.9     .07       0  5017.4     .05       0
  5036.4     .07       0
Bank Sta=5017.4,5036.4
XS Rating Curve= 0 ,0
Exp/Cntr=0.3,0.1

Type RM Length L Ch R = 1 ,37853   ,469,469,469
BEGIN DESCRIPTION:
BIG JOSHUA CREEK 68.0
END DESCRIPTION:
XS GIS Cut Line= 3
        2009675.       13869375.        2009675.       13869075.
        2009825.     13868724.99
#Sta/Elev= 30
    4700  1596.5    4740  1593.9    4760 1590.76    4810  1573.2    4830 1569.62
    4850 1567.23    4890 1564.52    4953 1562.91  5002.7 1563.91    5005 1553.22
  5005.5 1552.72  5024.1 1553.22  5050.4 1555.96  5061.7 1557.63  5085.2 1558.84
  5090.7 1561.19  5097.9 1562.03  5137.8 1563.03  5174.1 1562.94  5206.7 1562.27
  5219.4 1560.52  5228.5  1562.6  5237.5 1568.44    5272 1579.88  5282.9 1580.56
  5290.1 1582.33  5295.6 1580.43  5326.4 1585.72  5364.3 1589.26  5380.8 1590.15
#Mann= 6 ,-1 , 0
    4700     .12       0    4953    .035       0    5005    .035       0
  5024.1    .035       0  5050.4     .07       0  5364.3     .12       0
Bank Sta=5005,5024.1
XS Rating Curve= 0 ,0
Exp/Cntr=0.3,0.1

Type RM Length L Ch R = 1 ,37384   ,485,485,485
BEGIN DESCRIPTION:
BIG JOSHUA CREEK 67.0
END DESCRIPTION:
XS GIS Cut Line= 3
        2010125.     13869325.02        2010125.       13869125.
      2010082.96     13868363.48
#Sta/Elev= 30
    4800 1583.75    4830 1584.29    4870 1581.02    4920 1564.03    4930 1563.55
    4940 1560.39    4950 1552.98    4960 1551.63  4960.5 1549.34    4961 1548.84
  4979.6 1549.34  5002.1 1553.27  5030.1  1556.3  5050.1 1556.27  5070.1 1559.33
  5186.3 1560.64  5240.4 1561.58  5250.4 1563.48  5268.8 1572.02  5273.8 1569.71
  5280.4 1573.67  5310.5 1583.48  5330.5 1587.26  5383.7 1591.78  5449.6 1595.06
  5635.5  1600.4    5671 1605.55  5714.8 1606.81  5742.5 1607.13  5762.7 1607.51
#Mann= 8 ,-1 , 0
    4800     .12       0  4960.5     .05       0  4979.6     .12       0
  5002.1     .07       0  5186.3     .12       0  5383.7     .07       0
  5714.8     .12       0  5742.5     .07       0
Bank Sta=4960.5,4979.6
XS Rating Curve= 0 ,0
Exp/Cntr=0.3,0.1

Type RM Length L Ch R = 1 ,36899   ,423,423,423
BEGIN DESCRIPTION:
BIG JOSHUA CREEK 66.0
END DESCRIPTION:
XS GIS Cut Line= 3
      2010274.97     13869425.03        2010575.       13869125.
      2010835.38     13868785.95
#Sta/Elev= 30
  4571.3 1582.14  4627.9 1579.87  4691.2 1570.65  4810.3 1563.55  4821.9 1562.88
  4910.8 1559.21  4961.1 1549.43  4999.5  1545.7    5000  1545.2  5018.9  1545.7
  5031.9 1551.27  5067.2 1554.56  5085.7 1564.49  5102.5 1576.33  5117.1 1576.98
  5137.9 1585.12  5152.4 1587.44  5166.9 1579.49  5173.2 1584.71  5181.4 1578.28
  5187.7 1583.53  5202.2 1581.56  5216.8 1591.84  5223.1 1587.75  5260.3 1598.59
  5266.6 1594.12  5281.1  1603.4  5287.4 1601.83  5323.4 1614.18  5423.1 1623.81
#Mann= 8 ,-1 , 0
  4571.3    .035       0  4691.2     .07       0  4810.3     .12       0
  4821.9     .07       0  4961.1    .035       0  4999.5    .035       0
  5018.9    .035       0  5085.7     .12       0
Bank Sta=4999.5,5018.9
XS Rating Curve= 0 ,0
Exp/Cntr=0.3,0.1

Type RM Length L Ch R = 1 ,36476   ,458,458,458
BEGIN DESCRIPTION:
BIG JOSHUA CREEK 65.0
END DESCRIPTION:
XS GIS Cut Line= 3
       2010378.1     13869591.73        2010925.       13869325.
      2011074.99     13869175.01
#Sta/Elev= 30
  4391.3  1581.1  4476.6 1579.17  4512.6 1575.94  4535.1 1572.14  4557.6 1570.23
  4602.7 1568.19  4670.3 1567.26  4690.7 1565.64  4732.2  1561.7    4811 1558.96
  4850.5 1553.96  4873.1  1554.6  4918.1 1550.55  4923.7 1548.49  4929.3 1547.71
  4977.5 1546.26  4985.7 1545.45  4987.3 1543.42  4987.8 1542.92  5006.7 1543.42
  5013.7  1545.2  5042.2 1563.77  5056.3  1577.4  5070.5 1593.39  5084.6    1603
  5127.1 1629.28  5156.6  1634.6  5183.6 1637.73  5208.4 1642.92  5211.9 1642.92
#Mann= 9 ,-1 , 0
  4391.3    .035       0  4476.6     .07       0  4690.7    .035       0
  4732.2     .07       0  4929.3    .035       0  4987.3    .035       0
  5006.7    .035       0  5013.7     .07       0  5156.6     .12       0
Bank Sta=4987.3,5006.7
XS Rating Curve= 0 ,0
Exp/Cntr=0.3,0.1

Type RM Length L Ch R = 1 ,36018   ,393,393,393
BEGIN DESCRIPTION:
BIG JOSHUA CREEK 64.0
END DESCRIPTION:
XS GIS Cut Line= 3
      2010575.01       13869775.      2011092.36     13869701.04
      2011493.52     13869396.44
#Sta/Elev= 30
    4472 1578.02  4512.4  1576.5    4573 1565.42  4669.5    1562  4822.5 1558.44
  4922.5 1556.87  4936.7    1557  4987.2 1545.64  4993.4 1541.12  4998.8  1540.5
  4999.3    1540  5018.2  1540.5    5030 1541.67  5064.7 1544.43  5108.4 1558.72
  5114.6 1557.59  5122.9 1561.31  5128.3 1559.44  5143.7 1563.42    5150  1568.4
  5164.6 1573.61  5193.7 1580.71    5229 1585.73  5243.6 1591.46  5278.9 1594.54
  5336.9 1612.58  5393.3 1637.43  5436.9 1647.89  5443.2 1650.91  5498.3 1657.97
#Mann= 9 ,-1 , 0
    4472     .07       0  4669.5    .035       0  4822.5     .07       0
  4922.5    .035       0  4998.8    .035       0  5018.2    .035       0
    5030     .07       0  5128.3     .12       0  5436.9     .07       0
Bank Sta=4998.8,5018.2
XS Rating Curve= 0 ,0
Exp/Cntr=0.3,0.1

Type RM Length L Ch R = 1 ,35625   ,439,439,439
BEGIN DESCRIPTION:
BIG JOSHUA CREEK 63.0
END DESCRIPTION:
XS GIS Cut Line= 3
      2010386.75     13870056.14        2011125.       13870025.
      2011297.74     13870015.49
#Sta/Elev= 30
  4256.3 1578.74  4434.7 1576.26  4464.7  1573.8  4514.8 1571.84  4554.8 1568.15
  4564.8 1565.26  4584.8 1566.11  4624.9 1562.17  4694.9 1560.02    4815 1553.55
  4850.8 1553.15  4877.2 1553.12  4895.1    1553  4915.1 1548.82  4945.2 1547.59
  4955.2 1546.41  4965.2 1544.87  4979.9 1540.85  5015.5 1537.29    5016 1536.79
  5034.9 1537.29  5035.3 1539.59  5045.3 1545.44  5078.7 1574.79  5083.2 1579.25
  5088.3 1579.15  5105.4 1581.27  5145.4 1581.16  5164.3  1577.4  5168.2  1577.4
#Mann= 7 ,-1 , 0
  4256.3     .07       0  4850.8    .035       0  4877.2     .12       0
  4979.9    .035       0  5015.5    .035       0  5034.9    .035       0
  5078.7     .12       0
Bank Sta=5015.5,5034.9
XS Rating Curve= 0 ,0
Exp/Cntr=0.3,0.1

Type RM Length L Ch R = 1 ,35186   ,464,464,464
BEGIN DESCRIPTION:
BIG JOSHUA CREEK 62.0
END DESCRIPTION:
XS GIS Cut Line= 3
      2010824.95     13870374.99        2011025.       13870425.
        2011275.       13870425.
#Sta/Elev= 30
  4793.8 1573.14  4811.9 1573.91  4853.1 1572.56    4866  1571.1  4876.3 1567.74
  4886.6 1562.76  4894.3  1557.7  4898.5  1557.4  4917.5 1548.15  4927.9 1545.21
  4935.6 1541.43  4940.7  1541.5  4948.5 1538.48  4958.8 1536.63  4979.9 1536.07
  4980.4 1535.57  4999.4 1536.07    5020 1536.28    5030 1539.15  5034.9 1542.01
  5037.3 1543.41    5040 1544.98    5060 1549.26    5080 1549.64    5090 1548.52
    5100 1544.96    5120  1547.7    5200 1573.49    5230 1580.26    5250  1582.5
#Mann= 6 ,-1 , 0
  4793.8    .035       0  4898.5     .12       0  4979.9     .05       0
  4999.4     .12       0  5034.9    .035       0  5037.3     .12       0
Bank Sta=4979.9,4999.4
XS Rating Curve= 0 ,0
Exp/Cntr=0.3,0.1

Type RM Length L Ch R = 1 ,34722   ,584,584,584
BEGIN DESCRIPTION:
BIG JOSHUA CREEK 61.0
END DESCRIPTION:
XS GIS Cut Line= 3
      2010256.55     13871058.75        2011075.       13870875.
      2011325.01     13870774.99
#Sta/Elev= 30
  4156.9  1589.3  4354.3 1580.94  4370.5 1581.23    4426 1577.69  4462.8 1578.33
  4495.4 1576.53  4524.3 1574.88  4620.8 1573.44    4678 1573.49  4748.5 1568.81
  4800.6 1569.06  4836.4 1568.37  4862.5 1569.71  4923.1 1568.16  4954.7 1564.38
    4965 1559.35  4971.5 1550.27  4976.6 1548.36  4983.2 1532.19  4983.7 1531.69
  5003.1 1532.19  5040.2 1533.24    5059  1536.9  5071.1 1541.31  5081.9 1542.18
    5094 1545.38  5158.9 1552.42  5201.7 1558.97  5250.2 1568.94    5265 1570.72
#Mann= 9 ,-1 , 0
  4156.9     .12       0  4354.3    .035       0  4495.4     .07       0
  4620.8    .035       0  4748.5     .07       0  4800.6    .035       0
  4983.2    .035       0  5003.1    .035       0  5158.9     .12       0
Bank Sta=4983.2,5003.1
XS Rating Curve= 0 ,0
Exp/Cntr=0.3,0.1

Type RM Length L Ch R = 1 ,34138   ,571,571,571
BEGIN DESCRIPTION:
BIG JOSHUA CREEK 60.0
END DESCRIPTION:
XS GIS Cut Line= 3
      2010833.86     13871900.73        2011475.       13871275.
      2012275.03     13870474.97
#Sta/Elev= 30
  4108.8 1582.99  4293.2 1578.01  4629.8 1572.13  4799.6 1563.62  4842.6 1558.39
  4863.3 1558.65  4874.7 1555.12  4905.8 1541.91  4948.2 1530.88  4987.4 1530.18
  4987.9 1529.68  5007.8 1530.18    5033 1536.03    5040 1539.37  5047.1 1546.58
  5074.3 1551.44    5132 1555.84  5188.5 1563.33  5258.4 1563.11  5301.7 1565.98
  5400.7 1565.67  5527.9 1569.07  5598.7 1573.91  5626.9 1578.94  5655.2 1580.74
  5697.6 1588.38  5711.8 1588.51  5721.3 1591.24  6051.2 1657.31  6136.1 1678.74
#Mann= 9 ,-1 , 0
  4108.8     .12       0  4293.2     .07       0  4842.6    .035       0
  4874.7     .07       0  4987.4     .05       0  5007.8     .07       0
  5074.3     .12       0  5258.4    .035       0  5721.3     .12       0
Bank Sta=4987.4,5007.8
XS Rating Curve= 0 ,0
Exp/Cntr=0.3,0.1

Type RM Length L Ch R = 1 ,33567   ,583,583,583
BEGIN DESCRIPTION:
BIG JOSHUA CREEK 59.0
END DESCRIPTION:
XS GIS Cut Line= 3
      2011876.85     13871869.67        2011925.       13871525.
      2011958.79     13871022.25
#Sta/Elev= 30
    4652 1561.55  4761.7 1560.64  4878.9 1560.44    4899 1558.86  4909.1 1557.07
  4919.2 1552.56  4929.3 1544.93  4941.9 1533.91  4949.5 1527.66  4959.2 1527.29
  4979.7 1524.36  4980.2 1523.86  5000.1 1524.36  5002.5 1526.29  5020.1 1529.98
  5060.2 1536.87  5080.2 1539.08  5100.2 1539.73  5150.4 1544.01  5219.6 1551.56
  5224.6 1550.43  5230.5 1552.01  5250.6 1553.83  5266.7 1556.61  5280.6 1558.07
  5330.8 1558.79  5375.1 1561.51    5421 1562.16  5471.1 1565.33  5503.9 1565.04
#Mann= 8 ,-1 , 0
    4652     .12       0  4761.7     .07       0    4899    .035       0
  4941.9     .07       0  4979.7     .05       0  5000.1     .07       0
  5266.7     .12       0  5375.1    .035       0
Bank Sta=4979.7,5000.1
XS Rating Curve= 0 ,0
Exp/Cntr=0.3,0.1

Type RM Length L Ch R = 1 ,32984   ,560,560,560
BEGIN DESCRIPTION:
BIG JOSHUA CREEK 58.0
END DESCRIPTION:
XS GIS Cut Line= 3
        2012275.     13871874.99        2012475.       13871525.
        2012975.       13870725.
#Sta/Elev= 30
  4596.9 1556.69  4677.5 1556.86  4720.1 1553.53  4725.6    1553  4884.1 1532.38
  4911.5 1531.68  4934.1    1527  4997.5 1521.24    4998 1520.74  5017.9 1521.24
  5028.9 1523.61  5044.2 1542.07  5065.5 1550.98  5094.3 1556.25  5188.7 1562.54
  5295.5 1581.91  5348.5 1593.94  5369.7 1595.26  5479.4 1618.76  5500.6 1621.03
  5594.9 1649.54  5652.7 1670.43  5747.1 1711.03  5783.6 1728.74  5820.2 1751.64
    5878 1778.02  5914.5 1799.77  5935.7 1806.04  5940.5  1810.9  5943.4  1810.9
#Mann= 7 ,-1 , 0
  4596.9     .07       0  4720.1    .035       0  4725.6     .12       0
  4934.1     .07       0  4997.5     .05       0  5017.9     .07       0
  5295.5     .12       0
Bank Sta=4997.5,5017.9
XS Rating Curve= 0 ,0
Exp/Cntr=0.3,0.1

Type RM Length L Ch R = 1 ,32424   ,540,540,540
BEGIN DESCRIPTION:
BIG JOSHUA CREEK 57.0
END DESCRIPTION:
XS GIS Cut Line= 3
      2012474.96     13871975.01        2012875.       13871875.
        2013025.       13871075.
#Sta/Elev= 30
    4592 1556.14  4610.1 1555.84  4631.4 1552.52  4674.5  1544.1  4748.2 1538.68
  4849.7 1534.56  4898.7 1529.98  4932.2 1522.41  4963.2 1519.01  4963.7 1518.51
  4983.7 1519.01  5030.6 1521.59  5055.2 1530.33  5088.3 1547.04  5106.1 1550.93
  5140.9 1552.12  5187.5 1548.17  5251.1 1555.68  5340.1 1561.23    5399 1568.68
  5421.5 1574.14  5461.3 1580.09  5472.4  1583.6  5513.1 1588.83  5524.1 1592.64
  5563.9 1598.44  5629.2 1611.99  5635.2 1614.59  5739.4 1637.86  5818.3 1659.12
#Mann= 6 ,-1 , 0
    4592     .07       0  4631.4     .12       0  4748.2     .07       0
  4963.2     .05       0  4983.7     .07       0    5399     .12       0
Bank Sta=4963.2,4983.7
XS Rating Curve= 0 ,0
Exp/Cntr=0.3,0.1

Type RM Length L Ch R = 1 ,31884   ,549,549,549
BEGIN DESCRIPTION:
BIG JOSHUA CREEK 56.0
END DESCRIPTION:
XS GIS Cut Line= 3
      2012775.01       13872525.        2013125.       13872325.
      2013474.98     13872125.01
#Sta/Elev= 30
  4601.5 1548.55  4671.5 1546.93  4708.8 1543.05  4739.7 1538.27  4792.3 1533.97
  4916.1 1530.78  4931.9 1524.98    4947  1522.3  4953.5    1516  4959.3 1513.85
  4969.3 1510.93  4986.2 1509.85  4986.7 1509.35  5007.2 1509.85  5039.9  1516.6
    5050  1521.3  5055.7 1521.18  5077.3 1529.85  5093.1 1541.81  5108.3 1546.99
  5114.7 1550.52  5117.5 1549.92  5136.3 1551.08  5142.8 1553.62  5188.9 1553.56
  5201.1 1555.32  5232.8 1554.84  5291.8 1557.61  5327.1 1557.06  5407.7 1559.35
#Mann= 6 ,-1 , 0
  4601.5     .07       0  4671.5     .12       0  4708.8     .07       0
  4986.2     .05       0  5007.2     .07       0  5117.5     .12       0
Bank Sta=4986.2,5007.2
XS Rating Curve= 0 ,0
Exp/Cntr=0.3,0.1

Type RM Length L Ch R = 1 ,31335   ,537,537,537
BEGIN DESCRIPTION:
BIG JOSHUA CREEK 55.0
END DESCRIPTION:
XS GIS Cut Line= 3
      2012096.88     13872738.44        2013275.       13872825.
        2013475.       13872475.
#Sta/Elev= 30
  3818.7 1567.13  3979.4  1564.7  4127.6  1565.9  4167.8 1563.88  4227.9 1550.92
  4323.4 1548.01  4438.5 1542.68  4520.5 1543.65  4578.9 1546.22    4649 1544.77
  4661.5 1543.45  4709.2 1531.72  4829.5 1527.13  4909.8 1521.56  4933.3 1519.45
  4969.9 1506.95  4997.3 1506.83  4997.8 1506.33  5018.6 1506.83  5029.5 1507.02
  5035.3 1514.21  5066.9 1519.55  5072.7 1523.98  5088.5 1528.71  5094.3 1535.14
  5110.1 1537.44  5115.9    1542    5126 1543.47  5311.6  1545.4  5403.1 1547.67
#Mann= 6 ,-1 , 0
  3818.7     .12       0  4323.4    .035       0  4520.5     .12       0
  4997.3     .05       0  5018.6     .12       0  5311.6    .035       0
Bank Sta=4997.3,5018.6
XS Rating Curve= 0 ,0
Exp/Cntr=0.3,0.1

Type RM Length L Ch R = 1 ,30798   ,510,510,510
BEGIN DESCRIPTION:
BIG JOSHUA CREEK 54.0
END DESCRIPTION:
XS GIS Cut Line= 3
       2012448.4     13873888.61        2013525.       13873275.
        2013575.       13872875.
#Sta/Elev= 30
  3756.3 1583.97  3789.4 1582.12  3863.4 1579.23  3893.3 1578.11  4005.6 1573.08
  4013.7 1570.89  4019.4 1572.05  4051.2 1569.71  4078.5  1570.9  4284.4 1564.69
  4901.1 1549.32  4914.9 1544.54  4928.5 1532.19  4937.9 1530.26  4950.1 1523.67
  4960.2 1523.01  4972.5 1511.64  4981.8 1507.29  4993.5 1507.08  5027.7 1506.97
  5028.2 1506.47    5049 1506.97  5055.9 1509.85  5076.1 1511.18  5113.9 1522.78
  5194.5 1529.29  5280.2 1532.96    5318 1539.81  5346.6 1539.25  5398.6 1539.72
#Mann= 9 ,-1 , 0
  3756.3    .035       0  3789.4     .12       0  3863.4    .035       0
  3893.3     .07       0  4284.4    .035       0  4993.5     .12       0
  5027.7     .05       0    5049     .12       0  5346.6    .035       0
Bank Sta=5027.7,5049
XS Rating Curve= 0 ,0
Exp/Cntr=0.3,0.1

Type RM Length L Ch R = 1 ,30288   ,533,533,533
BEGIN DESCRIPTION:
BIG JOSHUA CREEK 53.0
END DESCRIPTION:
XS GIS Cut Line= 3
      2013825.01     13873724.97        2013975.       13873275.
      2013775.01     13872925.02
#Sta/Elev= 30
  4534.1 1560.97  4565.7 1559.52  4582.1 1556.07  4607.9 1549.37  4626.8 1549.14
  4660.6 1548.95  4681.6 1545.64  4692.4 1546.38  4702.7 1546.41  4734.4 1539.65
  4770.7 1537.81  4818.7 1535.01  4829.2 1532.95  4850.3 1533.85  4860.8 1528.53
  4881.9 1528.66  4892.5 1526.82  4913.5  1506.1  4945.2 1501.03  4976.7 1499.21
  4977.2 1498.71    4998 1499.21  5005.8 1503.92  5014.1  1505.3  5037.9 1509.86
  5081.1 1514.55  5118.6 1522.35  5220.8 1527.99  5274.5 1533.75  5411.5 1537.43
#Mann= 9 ,-1 , 0
  4534.1    .035       0  4582.1     .07       0  4626.8    .035       0
  4692.4     .07       0  4770.7    .035       0  4976.7    .035       0
    4998     .07       0  5014.1     .12       0  5274.5    .035       0
Bank Sta=4976.7,4998
XS Rating Curve= 0 ,0
Exp/Cntr=0.3,0.1

Type RM Length L Ch R = 1 ,29755   ,551,551,551
BEGIN DESCRIPTION:
BIG JOSHUA CREEK 52.0
END DESCRIPTION:
XS GIS Cut Line= 3
      2014149.81     13874044.83        2014475.       13873275.
      2014902.21     13872379.37
#Sta/Elev= 30
  4164.2 1563.59  4171.3 1563.47  4219.4 1561.99  4283.4 1559.24  4313.2 1552.87
  4478.8 1535.87  4696.4 1531.81  4885.1  1529.9  4902.2 1519.43  4908.8 1510.31
  4932.5 1502.08    4967 1499.38  4997.7 1499.29  4998.2 1498.79  5019.2 1499.29
  5022.1 1504.75  5031.2  1510.1  5073.8 1516.24  5150.2 1529.41  5218.3 1526.96
  5240.9 1522.79  5269.2 1509.41  5288.6 1519.97    5396  1543.2  5433.6 1551.14
  5553.9 1559.28  5841.6  1571.4  5932.5 1576.18  5938.7 1576.17  5992.2 1579.08
#Mann= 14 ,-1 , 0
  4164.2     .07       0  4171.3    .035       0  4219.4     .07       0
  4313.2    .035       0  4696.4     .07       0    4967    .035       0
  4997.7    .035       0  5019.2    .035       0  5073.8     .12       0
  5288.6    .035       0    5396     .07       0  5841.6     .12       0
  5932.5     .07       0  5938.7     .12       0
Bank Sta=4997.7,5019.2
XS Rating Curve= 0 ,0
Exp/Cntr=0.3,0.1

Type RM Length L Ch R = 1 ,29204   ,574,574,574
BEGIN DESCRIPTION:
BIG JOSHUA CREEK 51.0
END DESCRIPTION:
XS GIS Cut Line= 3
      2014625.01     13873624.99        2014975.       13873425.
      2015325.01     13872974.99
#Sta/Elev= 30
  4592.5 1528.26  4724.2 1526.57  4804.8 1519.05  4820.7 1519.21  4826.4 1517.48
  4901.3  1508.3  4907.1 1505.18  4998.8 1499.37  5006.3 1496.46  5006.8 1495.96
  5028.3 1496.46  5081.6 1496.88  5087.9 1499.44    5096 1513.46  5102.4 1513.48
  5109.6 1521.61  5122.6 1524.05  5145.8 1526.71    5173 1526.06  5251.7 1528.45
  5337.7 1533.07  5344.9 1534.99  5365.7 1536.58  5373.9 1539.59  5380.2 1540.14
  5409.1 1551.02    5430 1553.21  5473.4 1565.68  5539.2 1578.76  5565.7 1582.73
#Mann= 5 ,-1 , 0
  4592.5    .035       0  5006.3    .035       0  5028.3    .035       0
  5122.6     .12       0  5539.2     .07       0
Bank Sta=5006.3,5028.3
XS Rating Curve= 0 ,0
Exp/Cntr=0.3,0.1

Type RM Length L Ch R = 1 ,28630   ,515,515,515
BEGIN DESCRIPTION:
BIG JOSHUA CREEK 50.0
END DESCRIPTION:
XS GIS Cut Line= 3
      2015075.03     13873874.98        2015425.       13873675.
      2016074.96     13873125.03
#Sta/Elev= 30
  4591.9 1522.17  4826.9 1519.49  4914.4 1513.15  4943.9 1503.89  4949.6 1498.82
  5019.7 1496.55  5020.2 1496.05  5041.7 1496.55  5059.3 1496.65  5065.8 1503.64
  5073.9 1506.79    5182 1518.14  5335.6 1536.36  5349.3 1539.78  5371.3  1549.8
  5504.8 1569.13  5541.6 1572.36  5576.7 1584.41  5597.6 1586.33  5605.3 1582.84
  5611.8 1586.59  5619.6  1583.3  5626.1 1587.46  5633.9 1583.66  5640.4 1588.07
  5654.7 1591.53  5697.6 1616.95    5747  1633.1  5827.6 1650.77  5846.4 1652.75
#Mann= 8 ,-1 , 0
  4591.9     .07       0  4826.9    .035       0  5019.7    .035       0
  5041.7    .035       0  5073.9     .07       0    5182     .12       0
  5504.8     .07       0  5827.6     .12       0
Bank Sta=5019.7,5041.7
XS Rating Curve= 0 ,0
Exp/Cntr=0.3,0.1

Type RM Length L Ch R = 1 ,28115   ,559,559,559
BEGIN DESCRIPTION:
BIG JOSHUA CREEK 49.0
END DESCRIPTION:
XS GIS Cut Line= 3
      2015503.96     13874457.19        2015875.       13873875.
      2016125.01     13873174.98
#Sta/Elev= 30
  4309.6 1522.84  4352.8 1522.33  4800.9 1515.14  4898.4 1511.18  4928.8 1505.02
  4934.8 1498.59    4950 1492.24    4986 1488.93  4986.5 1488.43  5008.1 1488.93
  5035.3 1493.63  5084.9 1510.17  5134.8 1515.46  5138.6 1515.65  5405.1  1534.2
  5430.6 1546.29  5461.4 1552.79  5517.6 1574.69  5522.9 1573.26  5548.4  1588.3
  5553.7 1586.28  5566.6 1591.41  5579.2 1598.63  5584.5 1596.96  5604.7 1609.27
    5610 1607.65  5635.5 1624.79  5666.3 1637.58  5711.4 1650.08  5743.3 1652.62
#Mann= 9 ,-1 , 0
  4309.6    .035       0  4352.8     .07       0  4800.9    .035       0
    4986    .035       0  5008.1    .035       0  5035.3     .12       0
  5134.8     .07       0  5138.6     .12       0  5566.6     .07       0
Bank Sta=4986,5008.1
XS Rating Curve= 0 ,0
Exp/Cntr=0.3,0.1

Type RM Length L Ch R = 1 ,27556   ,522,522,522
BEGIN DESCRIPTION:
BIG JOSHUA CREEK 48.0
END DESCRIPTION:
XS GIS Cut Line= 3
      2015560.39     13874552.67        2016375.       13874075.
        2016375.     13873275.03
#Sta/Elev= 30
  4061.1  1523.3  4107.3 1522.44  4122.1 1522.71  4223.7 1518.84  4306.8 1514.58
  4355.4 1510.69  4522.7 1507.67  4559.9 1515.63  4676.1 1512.57  4686.4 1512.62
  4815.9 1512.99  4862.5 1508.77    4896 1502.81  4917.5 1491.05  4971.2  1487.2
  4971.7  1486.7  4993.3  1487.2  4995.8 1487.36  5035.4 1489.82  5085.4 1503.34
  5125.1 1507.88  5175.4 1510.77  5415.4 1513.22  5535.4 1519.12  5565.4 1522.99
  5605.4 1533.71  5655.4  1554.5  5725.4 1587.64  5755.4 1598.66  5805.4 1625.55
#Mann= 13 ,-1 , 0
  4061.1    .035       0  4107.3     .12       0  4122.1     .07       0
  4223.7     .12       0  4306.8     .07       0  4355.4     .12       0
  4676.1    .035       0  4686.4     .07       0  4862.5    .035       0
  4971.2     .05       0  4993.3    .035       0  4995.8     .07       0
  5125.1     .12       0
Bank Sta=4971.2,4993.3
XS Rating Curve= 0 ,0
Exp/Cntr=0.3,0.1

Type RM Length L Ch R = 1 ,27034   ,533,533,533
BEGIN DESCRIPTION:
BIG JOSHUA CREEK 47.0
END DESCRIPTION:
XS GIS Cut Line= 3
      2016625.02     13874574.97        2016825.       13874225.
      2017325.02     13873474.97
#Sta/Elev= 30
  4607.4 1509.04  4628.2 1508.65  4743.1    1505  4835.6 1503.26  4878.7 1499.67
  4906.8  1492.4  4921.9 1490.98  4929.9 1482.92  4947.9 1474.45  4948.4 1473.95
  4970.9 1474.45    5024  1475.8    5033 1482.08  5046.5 1485.08  5060.1 1493.42
  5069.1 1502.31  5110.1 1505.66  5321.6 1511.14  5427.3 1519.42  5501.7 1527.74
  5583.6 1542.86  5630.9 1559.51  5659.5 1562.58    5673 1568.11  5721.3 1572.72
  5745.1 1577.86  5796.2 1597.16  5839.8  1602.6  5889.3    1616  5911.9 1617.58
#Mann= 10 ,-1 , 0
  4607.4    .035       0  4628.2     .07       0  4743.1     .12       0
  4947.9     .05       0  4970.9     .12       0  5110.1     .07       0
  5321.6     .12       0  5427.3     .07       0  5583.6     .12       0
  5721.3     .07       0
Bank Sta=4947.9,4970.9
XS Rating Curve= 0 ,0
Exp/Cntr=0.3,0.1

Type RM Length L Ch R = 1 ,26501   ,540,540,540
BEGIN DESCRIPTION:
BIG JOSHUA CREEK 46.0
END DESCRIPTION:
XS GIS Cut Line= 3
      2016924.99     13874675.01        2017275.       13874475.
      2017474.98     13874125.03
#Sta/Elev= 30
  4592.3 1503.48  4651.4 1501.86  4739.9 1501.13  4766.9 1502.21  4783.1  1500.9
  4879.5 1499.85  4901.1 1496.24  4928.5 1484.67  4960.2 1482.04  4996.2 1473.71
  4997.6 1473.11  4998.1 1472.61  5020.7 1473.11    5053 1474.05  5062.4 1480.51
  5068.1 1488.69    5076 1495.96  5132.8 1508.62  5164.6 1519.65  5179.7 1521.55
  5207.8 1527.92  5223.6 1535.85  5237.3 1539.52  5282.6  1545.4  5288.4 1545.06
  5304.2 1551.36    5310  1550.7  5317.9 1554.27  5325.8  1555.8  5398.5  1559.1
#Mann= 7 ,-1 , 0
  4592.3     .07       0  4651.4    .035       0  4766.9     .12       0
  4996.2     .07       0  4997.6     .05       0  5020.7     .07       0
  5132.8     .12       0
Bank Sta=4997.6,5020.7
XS Rating Curve= 0 ,0
Exp/Cntr=0.3,0.1

Type RM Length L Ch R = 1 ,25961   ,564,564,564
BEGIN DESCRIPTION:
BIG JOSHUA CREEK 45.0
END DESCRIPTION:
XS GIS Cut Line= 3
      2016794.74     13875585.89        2017675.       13874775.
        2017825.     13874174.99
#Sta/Elev= 30
  3802.9 1538.25  3932.7 1532.06  3959.9 1530.74  4001.9 1529.46  4143.2  1518.5
  4284.9 1513.13  4355.8 1501.32  4454.9 1498.66    4738 1492.89  4773.2 1494.49
  4815.7 1493.29  4844.5 1489.87  4847.9 1489.71  4981.6 1471.03  4998.5 1469.92
    4999 1469.42  5021.6 1469.92  5022.9 1472.91  5051.3 1477.78    5059 1481.42
  5071.9 1505.77  5082.2 1511.66  5113.1 1513.27  5141.5 1509.54    5175 1508.24
  5218.5 1513.08  5371.6 1522.49  5566.6 1545.29    5595 1553.72  5618.2 1556.44
#Mann= 11 ,-1 , 0
  3802.9     .07       0  3932.7    .035       0  3959.9     .07       0
  4454.9    .035       0  4844.5     .12       0  4847.9    .035       0
  4981.6     .07       0  4998.5     .05       0  5021.6     .07       0
  5218.5     .12       0  5371.6     .07       0
Bank Sta=4998.5,5021.6
XS Rating Curve= 0 ,0
Exp/Cntr=0.3,0.1

Type RM Length L Ch R = 1 ,25397   ,540,540,540
BEGIN DESCRIPTION:
BIG JOSHUA CREEK 44.0
END DESCRIPTION:
XS GIS Cut Line= 4
      2017411.59     13875577.41        2017875.       13875275.
       2018074.1      13875144.3      2018228.72     13874794.58
#Sta/Elev= 30
    4442 1518.05  4496.7 1515.45  4505.1 1514.98  4511.1 1512.32  4526.2  1509.6
  4532.2 1506.45  4553.5 1502.47  4792.4 1490.52  4836.8 1486.17  4949.6 1476.71
  4959.5 1474.66  4972.7 1468.71  4976.1 1464.46  4976.6 1463.96  4999.5 1464.46
    5018 1467.59    5045 1480.89  5060.1 1491.89  5067.1  1494.6  5077.3 1495.11
  5111.4  1495.6  5155.9 1493.99  5288.9 1493.03  5397.6 1494.89  5451.4 1497.76
  5469.3 1502.04  5499.4 1506.65  5515.9 1509.36  5544.6 1511.04  5615.9 1513.38
#Mann= 10 ,-1 , 0
    4442    .035       0  4496.7     .07       0  4836.8     .12       0
  4976.1     .05       0  4999.5     .12       0  5077.3     .12       0
  5155.9     .07       0  5288.9    .035       0  5397.6     .07       0
  5499.4     .12       0
Bank Sta=4976.1,4999.5
XS Rating Curve= 0 ,0
Exp/Cntr=0.3,0.1

Type RM Length L Ch R = 1 ,24857   ,570,570,570
BEGIN DESCRIPTION:
BIG JOSHUA CREEK 43.0
END DESCRIPTION:
XS GIS Cut Line= 3
        2017625.       13875825.        2018075.       13875725.
      2018329.08     13874788.54
#Sta/Elev= 30
    4529 1535.52  4580.2 1531.44  4596.9 1526.35  4621.2 1521.91  4662.2 1517.26
  4689.1    1511  4694.2 1511.51  4754.4 1501.71  4815.8 1499.93  4838.3 1493.42
    4940 1479.93  4979.7 1476.31  5007.3 1467.25  5009.4 1463.35  5009.9 1462.85
  5032.8 1463.35  5081.8 1464.96  5093.6 1470.87  5121.6 1474.58  5136.4 1481.94
  5166.6 1489.49  5206.1 1491.53  5235.8 1492.94  5338.6 1491.74  5757.8 1491.83
  5818.9  1493.2    5847 1498.55  5852.2 1497.76  5886.8 1507.56  5960.3 1509.21
#Mann= 9 ,-1 , 0
    4529    .035       0  4838.3     .07       0    4940     .12       0
  5009.4     .05       0  5032.8     .12       0  5136.4     .07       0
  5206.1     .12       0  5338.6    .035       0  5757.8     .12       0
Bank Sta=5009.4,5032.8
XS Rating Curve= 0 ,0
Exp/Cntr=0.3,0.1

Type RM Length L Ch R = 1 ,24287   ,566,566,566
BEGIN DESCRIPTION:
BIG JOSHUA CREEK 42.0
END DESCRIPTION:
XS GIS Cut Line= 3
      2018375.01     13876424.98        2018525.       13875975.
      2018433.78     13874758.33
#Sta/Elev= 30
  4525.7 1520.66  4557.3 1517.86  4599.5 1506.53  4620.5 1498.22  4641.6 1492.83
  4797.2 1488.26  4872.3 1487.71    4908 1485.94  4926.2 1483.45  4936.8 1479.77
  4957.9 1467.58  4977.8 1458.71  4978.3 1458.21  5001.2 1458.71  5020.1 1461.58
  5040.1 1468.98  5050.2  1470.6  5090.3 1472.43  5100.3  1474.4  5120.4 1472.84
  5149.1 1475.35  5193.6 1479.79  5220.6  1484.7  5320.9 1487.94  5380.4 1487.31
  5591.7 1490.48  6052.8  1493.7  6137.5 1497.06  6183.3 1504.48  6220.1 1507.49
#Mann= 10 ,-1 , 0
  4525.7     .12       0  4797.2     .07       0  4872.3     .12       0
    4908     .07       0  4977.8     .05       0  5001.2     .07       0
  5149.1    .035       0  5193.6     .07       0  5380.4    .035       0
  6052.8     .12       0
Bank Sta=4977.8,5001.2
XS Rating Curve= 0 ,0
Exp/Cntr=0.3,0.1

Type RM Length L Ch R = 1 ,23721   ,550,550,550
BEGIN DESCRIPTION:
BIG JOSHUA CREEK 41.0
END DESCRIPTION:
XS GIS Cut Line= 3
      2018424.98     13876575.01        2019075.       13876025.
      2018802.58      13874669.9
#Sta/Elev= 30
  4148.5 1527.31  4184.2 1525.97  4212.8 1519.17  4276.5 1514.17  4311.7 1496.34
  4332.5 1489.69  4415.1 1484.58  4576.3 1482.64    4738 1484.29  4900.6 1481.53
  4957.7  1476.6    4972  1470.3  4978.6 1462.49  4998.4 1457.29  4998.9 1456.79
  5021.9 1457.29    5051 1458.87  5071.2 1464.55    5102 1463.51  5119.2 1469.55
  5223.8 1483.94  5321.2 1485.19  5324.2  1485.2  5527.4 1489.31  5807.8 1494.48
  6011.4  1495.2  6125.3 1495.21  6146.2 1495.16  6366.3 1501.76  6382.2  1503.2
#Mann= 14 ,-1 , 0
  4148.5     .12       0  4415.1     .07       0  4576.3    .035       0
  4998.4    .035       0  5021.9    .035       0  5119.2     .12       0
  5321.2    .035       0  5324.2     .07       0  5527.4    .035       0
  5807.8     .07       0  6011.4     .12       0  6125.3     .07       0
  6146.2     .12       0  6366.3     .07       0
Bank Sta=4998.4,5021.9
XS Rating Curve= 0 ,0
Exp/Cntr=0.3,0.1

Type RM Length L Ch R = 1 ,23171   ,1099,1099,1099
BEGIN DESCRIPTION:
BIG JOSHUA CREEK 40.0
END DESCRIPTION:
XS GIS Cut Line= 3
      2019077.81     13877152.77        2019575.       13876175.
      2019660.78     13876013.14
#Sta/Elev= 30
  3902.6 1526.94  4084.6 1523.94  4101.2 1521.42  4275.9 1514.55  4292.7 1511.63
  4301.5 1505.13  4315.2 1504.96  4323.7 1501.56  4329.3 1502.16    4346 1488.76
  4351.6 1486.77  4368.2 1476.09  4373.8 1475.58  4390.5 1468.16    4435 1470.32
  4567.3 1469.73  4594.4 1468.63  4663.1 1463.62  4718.6 1466.33  4793.1  1465.9
  4829.8 1465.09  4879.9 1459.94  4977.1 1458.13  4995.9 1453.26  4996.4 1452.76
  5019.4 1453.26  5022.2 1454.13  5035.3 1479.01  5131.3 1477.77  5182.7 1476.99
#Mann= 8 ,-1 , 0
  3902.6     .07       0  4275.9     .12       0  4567.3    .035       0
  4594.4     .12       0  4793.1     .07       0  4995.9     .05       0
  5019.4     .07       0  5131.3    .035       0
Bank Sta=4995.9,5019.4
XS Rating Curve= 0 ,0
Exp/Cntr=0.3,0.1

Type RM Length L Ch R = 1 ,22072   ,516,516,516
BEGIN DESCRIPTION:
BIG JOSHUA CREEK 39.0
END DESCRIPTION:
XS GIS Cut Line= 3
      2020140.39     13877066.97        2020025.       13876775.
      2019844.12     13876470.17
#Sta/Elev= 30
  4685.9 1501.51  4720.3  1503.1  4806.3 1505.29  4828.1 1505.43  4876.8 1504.15
  4882.2 1497.03  4892.3 1485.58  4901.2 1476.46  4903.6 1475.04  4906.5 1473.32
  4913.8 1465.55  4936.3 1451.58  4955.2 1448.81    4973 1448.22  4973.5 1447.72
  4996.4 1447.72  4996.9 1448.22  4997.2 1449.37  5002.8 1449.37  5013.5    1452
  5029.1 1453.74  5058.5 1460.01  5087.5 1460.02  5093.4 1461.04  5112.2 1460.72
  5204.5 1464.64  5225.9 1466.35  5255.7 1466.97  5305.8 1470.95  5354.3 1471.27
#Mann= 6 ,-1 , 0
  4685.9     .07       0  4903.6    .035       0    4973    .035       0
  4996.9    .035       0  5058.5     .07       0  5112.2    .035       0
Bank Sta=4973,4996.9
XS Rating Curve= 0 ,0
Exp/Cntr=0.3,0.1

Type RM Length L Ch R = 1 ,21556   ,527,527,527
BEGIN DESCRIPTION:
BIG JOSHUA CREEK 38.0
END DESCRIPTION:
XS GIS Cut Line= 3
      2020374.99     13876774.96        2020275.       13876375.
      2019501.38     13875173.36
#Sta/Elev= 30
  4581.9 1499.39  4734.2 1495.81  4829.2 1491.29  4847.3 1481.59  4852.4  1475.6
  4870.5 1463.04  4901.4 1447.41  4989.8  1445.7  4990.3  1445.2  5013.7  1445.7
  5046.5  1449.4    5125 1464.56  5192.6 1469.65  5724.7 1473.46  5767.2 1471.05
  5776.2 1467.86  5782.2 1470.36  5797.4 1463.23  5862.4 1462.66    5870 1467.83
  5872.7 1467.02  5875.9 1466.06  5885.2 1471.39  5906.3  1475.3  5992.1 1477.85
  6039.7 1481.36  6111.5 1484.69  6170.6 1486.99  6386.9 1490.67  6423.3 1492.41
#Mann= 12 ,-1 , 0
  4581.9     .07       0  4734.2    .035       0  4989.8    .035       0
  5013.7    .035       0  5046.5     .12       0  5192.6    .035       0
  5872.7     .07       0  5992.1     .12       0  6039.7     .07       0
  6111.5     .12       0  6170.6     .07       0  6386.9     .12       0
Bank Sta=4989.8,5013.7
XS Rating Curve= 0 ,0
Exp/Cntr=0.3,0.1
