HEC-RAS study BLOCK CREEK.prj: BLOCK CREEK Base Level Engineering

--- BLOCK CREEK.g01 (geometry) --- (continued)

Type RM Length L Ch R = 1 ,56138   ,462,462,462
BEGIN DESCRIPTION:
BLOCK CREEK 101.0
END DESCRIPTION:
XS GIS Cut Line= 3
        2011475.       13940575.        2011475.       13940225.
      2011324.99     13939624.96
#Sta/Elev= 30
  4650.4 1655.88  4690.4 1653.93  4733.1 1640.64  4760.4 1633.78  4834.3 1626.84
  4864.4 1623.63  4940.4 1622.65  5001.3 1615.22  5001.8 1614.72  5020.2 1615.22
  5024.3 1616.38  5051.9 1624.54    5271  1642.2  5307.1 1651.02  5312.2 1648.96
  5318.6 1652.58  5348.3 1664.11  5353.4 1662.26  5389.5  1680.9  5394.7 1678.86
  5430.7 1694.53  5435.9 1692.02    5472 1713.25  5477.1 1710.36  5513.2 1732.88
  5518.4 1730.77  5554.4 1752.17  5559.6 1750.64  5595.7 1766.51  5618.9 1770.43
#Mann= 8 ,-1 , 0
  4650.4     .05       0  4733.1    .035       0  4834.3     .07       0
  4864.4    .035       0  5001.3    .035       0  5020.2    .035       0
  5024.3     .07       0  5318.6     .12       0
Bank Sta=5001.3,5020.2
XS Rating Curve= 0 ,0
Exp/Cntr=0.3,0.1

Type RM Length L Ch R = 1 ,55676   ,459,459,459
BEGIN DESCRIPTION:
BLOCK CREEK 100.0
END DESCRIPTION:
XS GIS Cut Line= 3
        2011875.     13940425.04        2011875.       13940025.
      2011574.96     13939774.97
#Sta/Elev= 30
  4604.5 1643.88  4674.5 1633.32  4752.3 1629.67  4795.3 1628.57  4834.5 1627.83
  4874.5 1623.22  4894.5  1623.9  4924.5 1618.03  4954.5 1616.26  4964.5 1613.53
  4965.1 1610.48  4965.6 1609.98    4984 1610.48    5002 1616.99  5033.8 1617.86
    5069  1619.3  5075.5 1624.26  5096.3  1629.3  5196.5 1634.25  5210.9 1638.06
  5217.4 1642.98  5225.2 1644.69    5246 1652.69  5252.5 1656.83  5274.6 1664.31
  5303.3 1679.95  5309.8 1685.39  5338.4 1696.62  5367.1 1706.24  5395.1 1712.02
#Mann= 6 ,-1 , 0
  4604.5     .07       0  4752.3     .12       0  4795.3     .07       0
  4965.1     .05       0    4984     .07       0  5033.8     .12       0
Bank Sta=4965.1,4984
XS Rating Curve= 0 ,0
Exp/Cntr=0.3,0.1

Type RM Length L Ch R = 1 ,55217   ,481,481,481
BEGIN DESCRIPTION:
BLOCK CREEK 99.0
END DESCRIPTION:
XS GIS Cut Line= 3
       2012101.4     13940551.48        2012275.       13939875.
      2012074.99     13939274.96
#Sta/Elev= 30
  4301.1 1643.57  4369.7 1641.43  4456.9 1630.72  4524.6 1630.66  4602.1 1627.36
  4720.7 1625.51  4777.9 1618.98  4844.6 1618.55  4865.3 1615.71  4934.6  1613.3
  4981.7 1611.74  4987.4 1604.07  4987.9 1603.57  5006.4 1604.07    5010 1604.55
  5031.1 1620.13  5041.7 1623.82  5048.7 1624.19  5083.8 1624.37  5104.9 1627.89
  5147.1 1643.36  5199.8 1667.66  5294.6 1693.23  5336.8 1708.63  5357.9 1713.63
  5463.3 1749.26  5547.6 1770.71  5572.5 1779.53  5584.7 1784.32    5632 1800.66
#Mann= 8 ,-1 , 0
  4301.1     .07       0  4602.1     .12       0  4934.6     .07       0
  4987.4     .05       0  5006.4     .07       0  5048.7     .12       0
  5572.5     .07       0  5584.7     .12       0
Bank Sta=4987.4,5006.4
XS Rating Curve= 0 ,0
Exp/Cntr=0.3,0.1

Type RM Length L Ch R = 1 ,54736   ,436,436,436
BEGIN DESCRIPTION:
BLOCK CREEK 98.0
END DESCRIPTION:
XS GIS Cut Line= 3
      2012474.99     13940575.02        2012725.       13939975.
      2012674.99     13939774.98
#Sta/Elev= 30
  4353.9 1649.12  4363.1 1647.67  4397.8 1646.67  4416.2 1643.69  4429.8 1638.69
  4451.4 1633.39  4469.3 1631.33  4474.7  1628.8  4493.1 1625.35  4498.5 1622.55
  4551.6 1619.78  4594.4 1619.52  4668.1 1619.39  4787.8  1615.1  4835.5 1613.95
  4864.7 1614.74  4928.1 1612.19  4972.7 1602.28  4973.2 1601.78  4991.8 1602.28
  4994.7 1604.29  5001.2 1618.07  5006.5 1618.07  5014.2 1622.08    5022 1624.27
  5027.1  1623.5  5045.2 1626.31  5086.4 1626.56  5137.9 1628.95  5210.1 1633.95
#Mann= 4 ,-1 , 0
  4353.9     .07       0  4594.4     .12       0  4972.7     .05       0
  4991.8     .12       0
Bank Sta=4972.7,4991.8
XS Rating Curve= 0 ,0
Exp/Cntr=0.3,0.1

Type RM Length L Ch R = 1 ,54300   ,456,456,456
BEGIN DESCRIPTION:
BLOCK CREEK 97.0
END DESCRIPTION:
XS GIS Cut Line= 3
      2013174.99     13940774.96        2013075.       13940175.
      2012825.01     13939575.03
#Sta/Elev= 30
  4392.2 1713.23  4473.3 1697.55  4480.9 1694.48  4493.5 1684.73    4542  1661.3
  4552.7  1655.1  4574.6    1649  4602.5 1646.22    4676 1620.71  4696.3  1618.6
  4716.6 1619.91  4736.8 1615.39  4790.1 1612.68  4914.8 1611.01  4959.9 1604.82
  4980.2 1604.74  4988.3  1600.7  4988.8  1600.2  5007.4  1600.7  5032.9 1604.52
  5038.9 1607.95  5063.3 1608.54    5092 1611.33  5108.8 1615.81  5137.1 1615.58
  5213.2 1616.18  5368.8 1619.37    5508 1626.06  5617.9  1637.8  5650.4 1638.65
#Mann= 10 ,-1 , 0
  4392.2    .035       0    4542     .12       0  4552.7    .035       0
  4914.8     .07       0  4988.3     .05       0  5007.4     .07       0
  5063.3     .12       0  5137.1     .07       0  5213.2     .12       0
    5508     .07       0
Bank Sta=4988.3,5007.4
XS Rating Curve= 0 ,0
Exp/Cntr=0.3,0.1

Type RM Length L Ch R = 1 ,53844   ,429,429,429
BEGIN DESCRIPTION:
BLOCK CREEK 96.0
END DESCRIPTION:
XS GIS Cut Line= 3
      2013575.02     13940325.03        2013475.       13940125.
      2012874.98     13939524.98
#Sta/Elev= 30
  4771.6 1654.51    4808 1649.58  4824.7 1644.55  4847.1 1643.55  4883.4  1639.1
    4895 1638.77  4905.8 1637.71  4919.8  1633.2  4928.2 1632.68  4936.5 1627.48
  4942.1 1620.18  4950.5 1613.73  4958.9 1608.73  4964.5 1604.36  4972.9 1602.62
  4977.3 1597.61  4977.8 1597.11  4996.4 1597.61  5009.4 1598.68  5023.5 1603.92
    5066 1608.57  5094.2 1610.03  5122.5 1608.46  5142.2 1609.05  5433.6 1612.17
  5560.9 1616.36  5650.3 1621.56  5702.3 1624.37  5730.6 1626.79  5843.8  1639.5
#Mann= 6 ,-1 , 0
  4771.6    .035       0    4895     .07       0  4977.3     .05       0
  4996.4     .07       0  5142.2     .12       0  5650.3     .07       0
Bank Sta=4977.3,4996.4
XS Rating Curve= 0 ,0
Exp/Cntr=0.3,0.1

Type RM Length L Ch R = 1 ,53415   ,439,439,439
BEGIN DESCRIPTION:
BLOCK CREEK 95.0
END DESCRIPTION:
XS GIS Cut Line= 3
      2013822.85      13939780.2        2013575.       13939725.
      2012928.51     13939464.56
#Sta/Elev= 30
    4746 1630.94  4910.1 1631.96    4918 1631.63    4927 1628.06  4932.1 1627.58
  4938.4 1613.04  4945.8 1606.29  4948.7 1603.65  4966.1 1593.33  4966.6 1592.83
  4985.2 1593.33  4989.7 1593.55  4997.4 1598.72  5002.6 1598.72  5009.3 1600.85
  5014.7 1600.69  5021.5 1602.94  5032.3  1604.1  5056.9 1603.62  5129.3 1603.58
  5170.4 1605.45  5224.2 1606.22  5277.9 1609.09    5335 1610.74  5366.5 1613.57
  5390.7 1614.05  5463.2 1618.25  5544.9 1624.46  5551.8 1625.61  5696.9 1637.84
#Mann= 8 ,-1 , 0
    4746     .07       0  4910.1     .12       0  4945.8     .07       0
  4966.1     .05       0  4985.2     .07       0  5056.9     .12       0
    5335    .035       0  5544.9     .07       0
Bank Sta=4966.1,4985.2
XS Rating Curve= 0 ,0
Exp/Cntr=0.3,0.1

Type RM Length L Ch R = 1 ,52976   ,468,468,468
BEGIN DESCRIPTION:
BLOCK CREEK 94.0
END DESCRIPTION:
XS GIS Cut Line= 3
      2013878.88     13939388.16        2013625.       13939325.
      2013104.19     13939111.48
#Sta/Elev= 30
  4738.3 1624.05    4743 1624.05  4755.1 1624.18  4770.1 1624.35  4775.2 1623.33
  4793.8 1622.48    4835 1614.41  4852.7 1612.51  4935.4 1609.74  4948.4  1605.2
  4956.8  1603.3    4969 1600.55  4976.7 1597.53  4981.8 1597.05  4987.7 1592.61
  4988.2 1592.11  5006.9 1592.61  5014.6 1592.92  5060.1    1599  5097.4  1600.9
  5125.8 1604.25  5151.2 1607.52  5165.3 1607.89  5198.8 1608.15  5270.5 1611.83
  5358.9 1617.04  5412.3  1622.6  5425.3  1625.2  5475.5 1628.91  5562.8 1640.79
#Mann= 11 ,-1 , 0
  4738.3     .12       0    4743     .07       0  4755.1     .12       0
  4956.8     .07       0  4987.7     .05       0  5006.9     .07       0
  5060.1    .035       0  5125.8     .07       0  5165.3    .035       0
  5270.5     .07       0  5425.3    .035       0
Bank Sta=4987.7,5006.9
XS Rating Curve= 0 ,0
Exp/Cntr=0.3,0.1

Type RM Length L Ch R = 1 ,52508   ,457,457,457
BEGIN DESCRIPTION:
BLOCK CREEK 93.0
END DESCRIPTION:
XS GIS Cut Line= 3
      2013975.01     13939125.01        2013725.       13938925.
        2013425.     13938475.01
#Sta/Elev= 30
  4679.8 1619.83  4707.8 1617.76  4729.6 1612.28  4751.1 1608.23  4815.1 1606.24
  4850.3 1599.81  4879.1 1600.95  4914.3 1597.12  4949.6 1597.26  5018.9 1590.53
  5019.4 1590.03  5038.1 1590.53  5049.6 1601.29  5064.6  1609.6  5100.6 1611.93
  5144.2 1619.34  5172.7 1621.37  5229.8 1631.45  5284.3 1644.24    5317 1655.49
    5353 1663.33  5383.1 1679.34  5389.1 1680.58  5404.1 1691.89  5440.2 1711.56
  5461.6 1719.48  5468.7 1723.93  5518.3 1742.37    5525 1742.89  5540.8 1744.13
#Mann= 7 ,-1 , 0
  4679.8     .12       0  4729.6     .07       0  5018.9     .05       0
  5038.1     .07       0  5284.3     .12       0  5461.6     .07       0
    5525     .12       0
Bank Sta=5018.9,5038.1
XS Rating Curve= 0 ,0
Exp/Cntr=0.3,0.1

Type RM Length L Ch R = 1 ,52051   ,380,380,380
BEGIN DESCRIPTION:
BLOCK CREEK 92.0
END DESCRIPTION:
XS GIS Cut Line= 3
        2014075.     13939024.99        2014075.       13938675.
      2013354.76     13938087.43
#Sta/Elev= 30
  4644.7 1613.37  4694.7 1611.55  4744.7 1603.98  4884.7 1600.27  4984.7 1590.89
  4998.7 1584.92  4999.2 1584.42    5018 1584.92  5051.4 1597.97  5129.7 1614.89
  5193.6 1606.84  5207.9 1616.97  5222.3 1621.87    5307 1642.75  5329.3 1653.38
  5356.6 1656.48  5393.2 1671.51  5399.7 1670.23  5407.6 1677.36    5414 1676.65
  5428.4 1695.03  5471.5 1705.69  5591.4 1716.11  5648.8 1730.64    5684 1731.81
  5698.4 1738.51  5712.7 1740.19  5854.4 1745.82  5916.2 1749.88  5924.2 1748.98
#Mann= 5 ,-1 , 0
  4644.7     .07       0  4998.7     .05       0    5018     .07       0
  5854.4    .035       0  5916.2     .07       0
Bank Sta=4998.7,5018
XS Rating Curve= 0 ,0
Exp/Cntr=0.3,0.1

Type RM Length L Ch R = 1 ,51671   ,509,509,509
BEGIN DESCRIPTION:
BLOCK CREEK 91.0
END DESCRIPTION:
XS GIS Cut Line= 3
      2014370.46     13938929.59      2014403.56     13938518.84
      2014292.61     13937828.27
#Sta/Elev= 30
  4593.8 1602.69  4678.7 1601.49  4761.5 1599.94  4869.3 1598.84  4963.1 1589.04
  4979.6 1586.31    4980 1582.94  4980.5 1582.44  4999.3 1582.94    5014 1588.45
  5026.6 1594.87  5060.4 1603.16  5088.6 1614.45  5093.6 1619.71    5111 1624.53
  5171.8  1656.9  5192.1 1675.47  5202.2 1680.72  5209.3 1681.09  5222.5 1684.25
  5273.1 1685.02  5293.4 1690.28  5341.2 1692.93  5346.3 1696.37  5374.4 1701.86
  5455.4 1709.99  5502.9 1719.95  5576.9 1731.74  5607.3 1740.99  5705.3 1756.13
#Mann= 8 ,-1 , 0
  4593.8    .035       0  4678.7     .07       0  4761.5    .035       0
    4980    .035       0  4999.3    .035       0    5014     .12       0
  5209.3     .07       0  5502.9    .035       0
Bank Sta=4980,4999.3
XS Rating Curve= 0 ,0
Exp/Cntr=0.3,0.1

Type RM Length L Ch R = 1 ,51162   ,470,470,470
BEGIN DESCRIPTION:
BLOCK CREEK 90.0
END DESCRIPTION:
XS GIS Cut Line= 3
      2014425.02     13938924.98        2014825.       13938625.
        2014975.       13938475.
#Sta/Elev= 30
  4495.2 1601.69  4595.2 1599.81  4637.9 1599.85    4667 1598.34  4687.9  1598.9
  4702.5 1598.18    4717 1598.88  4723.3 1597.71    4767 1597.84  4837.9  1595.3
  4887.9 1591.94  4945.2 1591.65  4952.5 1591.14    4967 1588.46  4987.9 1585.77
    4992 1583.76  4998.7 1583.76  4999.7 1581.32  5000.2 1580.82  5018.5 1580.82
    5019 1581.32  5023.5 1582.06  5064.1 1597.79    5080 1606.13  5094.2 1615.22
  5123.3  1631.8  5150.7 1645.95  5164.9 1650.14  5203.8 1658.36  5207.3 1658.36
#Mann= 5 ,-1 , 0
  4495.2    .035       0  4999.7    .035       0    5019    .035       0
  5064.1     .07       0  5123.3     .12       0
Bank Sta=4999.7,5019
XS Rating Curve= 0 ,0
Exp/Cntr=0.3,0.1

Type RM Length L Ch R = 1 ,50692   ,444,444,444
BEGIN DESCRIPTION:
BLOCK CREEK 89.0
END DESCRIPTION:
XS GIS Cut Line= 3
      2014574.97     13939425.02        2015175.       13938925.
      2015375.01     13938574.98
#Sta/Elev= 30
  4218.7 1608.97  4254.5 1608.42  4310.5  1600.6  4885.9 1589.81    4908 1585.02
  4921.7  1585.7  4943.1 1582.74  4986.8 1581.33  4987.3 1580.83  5006.2 1581.33
    5035 1587.97  5045.1 1588.69  5050.9 1591.61  5066.7 1589.95  5072.5 1592.44
  5088.3 1590.42  5094.1 1593.37  5109.9 1590.96  5131.5 1599.13  5147.3 1602.13
  5153.1 1604.83  5168.9  1605.5  5174.7 1609.07    5192 1610.22  5196.3 1613.57
    5210 1615.84  5233.7    1620  5321.3 1645.12  5367.6 1655.11  5402.9 1659.23
#Mann= 6 ,-1 , 0
  4218.7    .035       0  4986.8    .035       0  5006.2    .035       0
    5192     .07       0    5210     .12       0  5321.3     .07       0
Bank Sta=4986.8,5006.2
XS Rating Curve= 0 ,0
Exp/Cntr=0.3,0.1

Type RM Length L Ch R = 1 ,50248   ,470,470,470
BEGIN DESCRIPTION:
BLOCK CREEK 88.0
END DESCRIPTION:
XS GIS Cut Line= 3
      2014874.96     13939525.02        2015425.       13939275.
      2015525.02     13939024.96
#Sta/Elev= 30
  4395.8 1599.16  4593.6 1595.74  4605.7 1594.82  4669.4 1592.67  4681.4 1591.75
  4824.2 1587.86  4857.2 1587.18  4934.1 1587.01    4941 1585.39  4956.1 1581.56
  4962.7 1581.01    4978 1580.95  4981.5 1578.75    4982 1578.25  5000.4 1578.25
  5000.9 1578.75  5063.3 1582.25  5068.7 1584.36  5086.2  1588.4  5098.3 1592.53
  5117.1  1594.4  5122.5 1595.61  5143.2 1596.01  5193.9 1601.26  5200.6 1602.71
    5206  1603.2  5224.8 1607.41  5236.9 1611.01  5259.8  1614.8  5269.3 1614.82
#Mann= 5 ,-1 , 0
  4395.8    .035       0    4941     .07       0  4981.5     .05       0
  5000.9     .07       0  5143.2     .12       0
Bank Sta=4981.5,5000.9
XS Rating Curve= 0 ,0
Exp/Cntr=0.3,0.1

Type RM Length L Ch R = 1 ,49778   ,535,535,535
BEGIN DESCRIPTION:
BLOCK CREEK 87.0
END DESCRIPTION:
XS GIS Cut Line= 3
      2015175.03     13940174.97        2015725.       13939625.
      2015827.09     13939284.13
#Sta/Elev= 30
    4227 1632.99  4283.5 1628.64    4333 1619.71  4354.2 1617.28  4437.8 1610.09
  4477.2  1607.4  4566.4 1598.98  4634.4 1596.49  4707.8  1593.2  4806.8 1591.93
  4820.9 1590.12  4877.5 1587.95  4905.8 1580.36  4925.4 1578.01  4926.4 1577.99
  4962.3 1576.58  4976.5 1572.91  4980.9 1572.76  4981.4 1572.26  5000.4 1572.76
  5001.2 1576.83  5017.2 1577.37  5036.1 1577.52  5046.5 1578.62  5059.6 1582.19
  5109.2 1585.78  5125.8 1588.28  5197.2  1588.8  5292.8 1592.61  5360.6 1594.85
#Mann= 10 ,-1 , 0
    4227     .07       0  4437.8    .035       0  4477.2     .07       0
  4634.4    .035       0  4925.4     .07       0  4926.4    .035       0
  4980.9    .035       0  5000.4    .035       0  5017.2     .07       0
  5292.8    .035       0
Bank Sta=4980.9,5000.4
XS Rating Curve= 0 ,0
Exp/Cntr=0.3,0.1

Type RM Length L Ch R = 1 ,49243   ,585,585,585
BEGIN DESCRIPTION:
BLOCK CREEK 86.0
END DESCRIPTION:
XS GIS Cut Line= 3
      2016324.99     13940224.99        2016125.       13939875.
        2015775.     13939075.01
#Sta/Elev= 30
  4596.9 1612.69  4700.5 1606.19  4750.2 1598.52  4793.4  1596.7  4803.5 1597.88
  4815.7 1596.83  4846.7 1597.08  4905.7 1593.72  4911.5 1592.13  4948.9 1591.83
  4964.7 1585.88  4970.5 1581.97    4977 1575.07  4997.1 1567.54  5021.3 1566.13
  5021.8 1565.63  5043.5 1566.13  5043.7 1571.62  5054.6 1574.71  5066.7 1576.24
  5081.2    1576  5113.4 1576.83  5142.3 1579.76  5152.8 1578.77  5244.6 1583.24
  5353.4 1585.28  5637.4 1593.44  5730.9 1598.34  5818.4 1604.63  5873.2 1609.17
#Mann= 7 ,-1 , 0
  4596.9     .07       0  5021.3     .05       0  5043.5     .07       0
  5081.2     .12       0  5244.6     .07       0  5353.4    .035       0
  5818.4     .07       0
Bank Sta=5021.3,5043.5
XS Rating Curve= 0 ,0
Exp/Cntr=0.3,0.1

Type RM Length L Ch R = 1 ,48658   ,586,586,586
BEGIN DESCRIPTION:
BLOCK CREEK 85.0
END DESCRIPTION:
XS GIS Cut Line= 3
      2016645.26     13939691.34        2016475.       13939425.
      2016221.22     13939119.72
#Sta/Elev= 30
  4684.1 1604.96  4841.2 1601.44  4881.9 1596.97  4898.7 1593.55  4905.3 1590.29
    4929 1581.12  4935.1 1578.05    4941 1576.86  4950.3  1572.4  4964.6 1569.05
  4971.4 1567.05  4977.4 1564.51  4981.5  1564.2    4982  1563.7  5003.2  1563.7
  5003.7  1564.2  5007.4 1564.44  5013.9 1570.14  5021.7 1571.48  5050.3 1570.61
  5056.8 1571.18  5078.2 1570.59    5092  1573.1  5095.1 1574.47  5106.3 1578.77
  5128.5 1582.52    5135 1582.88  5156.3 1582.37  5319.9 1584.71  5397.2 1587.04
#Mann= 5 ,-1 , 0
  4684.1     .07       0  4881.9     .12       0  4981.5     .05       0
  5003.7     .12       0  5095.1    .035       0
Bank Sta=4981.5,5003.7
XS Rating Curve= 0 ,0
Exp/Cntr=0.3,0.1

Type RM Length L Ch R = 1 ,48072   ,558,558,558
BEGIN DESCRIPTION:
BLOCK CREEK 84.0
END DESCRIPTION:
XS GIS Cut Line= 3
      2017048.22     13939268.42        2016875.       13939025.
      2016684.12     13938785.53
#Sta/Elev= 30
    4701 1583.57  4745.9 1582.99  4906.3 1578.33  4921.1 1575.32    4942 1567.16
  4969.9 1565.62  4977.6 1564.52  4985.5 1560.33    4986 1559.83  5007.8 1560.33
  5013.4 1563.09  5027.8 1564.07  5035.8 1562.93    5047 1565.45  5050.2 1566.64
    5071 1566.33  5135.1 1574.13  5191.6 1578.91  5219.9 1585.93    5228  1591.1
  5234.4 1592.02  5242.4 1598.64  5248.8 1599.67  5255.5 1606.65  5263.2 1611.34
    5284 1613.39    5292 1615.42  5298.4  1614.6  5303.1  1617.6    5306  1617.6
#Mann= 6 ,-1 , 0
    4701     .07       0  4745.9     .12       0  4969.9    .035       0
  4985.5    .035       0  5007.8    .035       0    5047     .12       0
Bank Sta=4985.5,5007.8
XS Rating Curve= 0 ,0
Exp/Cntr=0.3,0.1

Type RM Length L Ch R = 1 ,47514   ,530,530,530
BEGIN DESCRIPTION:
BLOCK CREEK 83.0
END DESCRIPTION:
XS GIS Cut Line= 3
      2017575.01     13939125.01        2017325.       13938725.
      2016925.01     13938575.01
#Sta/Elev= 30
  4532.9 1587.16  4561.8 1586.12  4611.3 1573.33  4692.7 1568.86  4902.6 1568.43
  4923.8 1566.95  4945.7 1562.16  4969.2  1562.6  4988.8 1558.29  5003.3  1556.5
  5003.8    1556  5025.6  1556.5    5026 1559.43  5034.4 1560.77  5080.3 1564.14
  5165.7 1579.51  5185.3 1581.39  5196.9 1589.81  5215.5 1593.23  5220.9 1597.67
  5245.8  1605.7  5251.1  1609.9  5270.7 1612.39  5282.3 1618.79    5301 1622.28
  5314.3 1627.61  5363.1  1637.1  5411.6 1654.67  5416.7 1657.64  5431.8 1659.07
#Mann= 8 ,-1 , 0
  4532.9     .07       0  4611.3    .035       0  4988.8     .07       0
  5003.3     .05       0  5025.6     .07       0  5034.4     .12       0
  5363.1     .07       0  5411.6    .035       0
Bank Sta=5003.3,5025.6
XS Rating Curve= 0 ,0
Exp/Cntr=0.3,0.1

Type RM Length L Ch R = 1 ,46984   ,564,564,564
BEGIN DESCRIPTION:
BLOCK CREEK 82.0
END DESCRIPTION:
XS GIS Cut Line= 3
        2017875.     13939075.04        2017825.       13938625.
      2017374.99     13937974.98
#Sta/Elev= 30
  4546.7 1588.62  4556.8 1588.54  4602.1 1567.82  4607.1 1566.35  4701.4 1564.38
    4900 1561.31  4964.8 1557.85  4989.5 1554.99  5002.6 1556.44  5010.6 1554.74
  5011.1 1554.24    5033 1554.74    5036 1557.01  5072.5  1557.2  5084.7 1559.48
  5099.5 1567.76  5121.5 1573.16  5275.1 1580.01    5382 1587.37  5466.4  1602.7
    5538 1620.95  5573.9 1625.56  5595.5 1633.08  5609.7 1635.47  5654.1  1648.3
  5696.2 1660.78  5753.6 1689.85  5764.8 1692.55  5779.8 1694.57  5790.1 1695.17
#Mann= 13 ,-1 , 0
  4546.7     .12       0  4602.1     .07       0  4701.4    .035       0
    4900     .12       0  4964.8    .035       0  5010.6    .035       0
    5033    .035       0  5121.5     .07       0  5275.1    .035       0
    5382     .07       0  5654.1     .12       0  5764.8     .07       0
  5779.8     .12       0
Bank Sta=5010.6,5033
XS Rating Curve= 0 ,0
Exp/Cntr=0.3,0.1

Type RM Length L Ch R = 1 ,46420   ,579,579,579
BEGIN DESCRIPTION:
BLOCK CREEK 81.0
END DESCRIPTION:
XS GIS Cut Line= 4
      2018296.73     13939252.47        2018325.       13938825.
      2018295.49     13938580.57      2018084.09     13938356.32
#Sta/Elev= 30
    4572 1586.29  4599.5 1584.17  4649.6 1584.14  4729.8  1581.9  4749.9 1580.26
  4789.1 1578.91  4791.2 1578.87    4820 1578.92  4840.1 1576.24  4860.1 1568.55
  4870.1 1563.48  4889.5  1556.6  4910.2 1552.47  4919.9 1554.01  4924.9 1553.11
  4940.3 1553.74  4986.7 1548.21  4987.2 1547.71  5009.2 1548.21  5010.5 1549.56
  5020.6  1551.5  5043.9 1553.23  5060.8 1558.51  5091.1 1557.01  5161.6 1559.35
  5186.6 1559.34  5301.9 1560.34  5345.1 1560.79  5399.5 1561.71  5554.8 1566.82
#Mann= 9 ,-1 , 0
    4572    .035       0  4789.1     .07       0  4791.2     .12       0
  4889.5     .07       0  4986.7     .05       0  5009.2     .07       0
  5186.6    .035       0  5301.9     .07       0  5345.1     .12       0
Bank Sta=4986.7,5009.2
XS Rating Curve= 0 ,0
Exp/Cntr=0.3,0.1

Type RM Length L Ch R = 1 ,45841   ,539,539,539
BEGIN DESCRIPTION:
BLOCK CREEK 80.0
END DESCRIPTION:
XS GIS Cut Line= 3
      2019255.88     13938539.47        2018725.       13938525.
      2018203.33     13938363.41
#Sta/Elev= 30
    4469 1581.34  4489.9  1578.4  4519.9 1576.43  4529.9 1573.66  4539.9 1574.69
  4610.6 1570.68    4730 1566.53  4807.6 1566.09    4870  1564.5    4880 1562.82
  4906.2 1561.03    4920 1556.49    4930 1551.26  4957.7 1543.97  4958.2 1543.47
  4982.4 1543.97  5002.7 1544.02  5021.6 1546.01    5042 1544.55  5062.9 1550.16
  5086.8 1551.11  5114.2 1553.86  5184.6 1556.65  5215.1 1556.79  5257.2 1556.41
  5419.4 1558.26  5461.1 1559.45  5471.2 1561.05    5516  1561.8  5546.2 1562.79
#Mann= 10 ,-1 , 0
    4469     .12       0  4610.6    .035       0  4807.6     .07       0
  4906.2     .12       0  4957.7     .05       0  4982.4     .12       0
  5215.1    .035       0  5257.2     .12       0  5419.4    .035       0
    5516     .12       0
Bank Sta=4957.7,4982.4
XS Rating Curve= 0 ,0
Exp/Cntr=0.3,0.1

Type RM Length L Ch R = 1 ,45302   ,545,545,545
BEGIN DESCRIPTION:
BLOCK CREEK 79.0
END DESCRIPTION:
XS GIS Cut Line= 3
      2019067.44      13938046.6        2018675.       13938025.
       2017949.6     13937989.44
#Sta/Elev= 30
  4606.6  1558.4  4756.9 1558.28  4839.4 1558.86  4889.5 1544.73  4929.5  1539.5
  4959.6  1543.2  4979.6 1540.94  4984.7  1537.6  4985.2  1537.1  5009.5  1537.6
  5029.7 1545.28  5059.7 1545.71  5098.3 1550.46  5129.8 1546.85  5169.8  1548.4
  5189.9 1545.49  5209.9 1548.73  5263.2  1551.6    5280 1555.01    5300 1562.69
  5318.8 1561.52  5380.1 1561.04  5409.1 1567.92  5460.2 1579.16  5488.2 1580.91
  5507.8 1580.24  5512.8 1582.26  5613.8 1588.56  5700.5 1593.41  5725.9 1600.52
#Mann= 9 ,-1 , 0
  4606.6    .035       0  4756.9     .12       0  4984.7     .05       0
  5009.5     .12       0  5263.2     .07       0  5318.8     .12       0
  5409.1     .07       0  5488.2    .035       0  5613.8     .07       0
Bank Sta=4984.7,5009.5
XS Rating Curve= 0 ,0
Exp/Cntr=0.3,0.1

Type RM Length L Ch R = 1 ,44757   ,571,571,571
BEGIN DESCRIPTION:
BLOCK CREEK 78.0
END DESCRIPTION:
XS GIS Cut Line= 3
      2019222.71     13937730.86        2018625.       13937525.
      2018242.55     13937377.41
#Sta/Elev= 30
  4367.4 1559.19  4660.7 1548.28  4827.9 1547.22    4867 1544.35  4904.4 1542.08
  4936.1 1535.25  4967.8 1535.66  4976.8 1532.77  4977.3 1532.27  5001.7 1532.77
  5002.2 1534.34  5014.5 1533.12  5044.5    1536  5069.1 1535.63  5093.7 1539.81
  5117.5 1551.45    5129    1561  5148.3 1570.61  5160.3 1584.85  5202.9 1597.79
  5208.2 1601.53  5232.8 1605.51  5238.2 1609.58  5268.2 1612.25  5287.4 1607.24
  5317.4  1607.7  5322.7  1610.8    5342 1608.99  5387.5 1616.21  5409.5 1619.24
#Mann= 6 ,-1 , 0
  4367.4    .035       0  4660.7     .12       0    4867     .07       0
  4976.8     .05       0  5001.7     .07       0  5387.5     .12       0
Bank Sta=4976.8,5001.7
XS Rating Curve= 0 ,0
Exp/Cntr=0.3,0.1

Type RM Length L Ch R = 1 ,44186   ,1132,1132,1132
BEGIN DESCRIPTION:
BLOCK CREEK 77.0
END DESCRIPTION:
XS GIS Cut Line= 3
      2019274.99     13937324.99        2018925.       13937075.
      2018525.02     13936875.01
#Sta/Elev= 30
  4565.3 1554.72  4614.4 1552.62  4658.7 1545.43  4700.5 1541.88  4795.1 1541.32
  4872.5 1536.13  4922.9 1535.91  4958.5 1528.37  4991.3 1526.68  4991.8 1526.18
  5016.3 1526.68  5026.2 1531.64  5054.1 1536.97  5070.9 1549.83  5093.2 1562.12
  5098.8 1560.18  5115.6 1564.81  5121.2 1563.95    5138 1570.26  5143.5 1569.63
  5155.8 1577.36  5200.2 1589.15  5210.6 1590.98  5227.4 1599.35  5249.8 1606.64
  5294.5 1615.58  5308.5  1616.3  5330.8 1625.87    5401 1647.35  5442.6 1658.54
#Mann= 6 ,-1 , 0
  4565.3     .12       0  4991.3     .05       0  5016.3     .12       0
  5155.8    .035       0  5200.2     .07       0    5401     .12       0
Bank Sta=4991.3,5016.3
XS Rating Curve= 0 ,0
Exp/Cntr=0.3,0.1

Type RM Length L Ch R = 1 ,43460   ,406,406,406
BEGIN DESCRIPTION:
BLOCK CREEK 76.0
END DESCRIPTION:
XS GIS Cut Line= 3
      2019811.65     13937097.29      2019444.84     13936654.62
      2019025.03     13936125.03
#Sta/Elev= 30
  4425.1  1565.6  4547.5 1554.37  4587.4 1549.78  4729.4 1547.73  4783.2 1545.44
  4815.4 1543.02  4879.2 1529.57  4928.6 1529.04  4971.6 1526.17  4973.4 1524.15
  4973.9 1523.65  4998.6 1524.15  5056.5 1530.98  5077.3 1537.48  5091.8 1539.71
    5191 1545.59  5312.9  1556.5  5356.2 1561.28  5369.6 1564.18  5391.4 1575.26
  5426.7 1586.09  5461.9 1602.25  5484.4 1609.75  5505.2 1616.32  5548.2 1626.53
  5590.1 1641.33    5612 1646.28  5633.4 1654.09  5662.2 1660.24  5675.8 1661.08
#Mann= 6 ,-1 , 0
  4425.1     .12       0  4547.5     .07       0  4783.2     .12       0
  4973.4     .05       0  4998.6     .12       0    5191     .07       0
Bank Sta=4973.4,4998.6
XS Rating Curve= 0 ,0
Exp/Cntr=0.3,0.1

Type RM Length L Ch R = 1 ,43054   ,552,552,552
BEGIN DESCRIPTION:
BLOCK CREEK 75.0
END DESCRIPTION:
XS GIS Cut Line= 3
        2019925.       13936975.        2019775.       13936525.
      2019124.99     13935824.99
#Sta/Elev= 30
  4525.1 1560.52  4567.3 1558.31  4583.2 1555.04  4630.5 1550.18  4732.1 1547.92
  4792.7  1546.3  4897.5 1543.67  4915.1 1539.46  4936.2 1528.87  4957.3 1526.44
  4965.7 1521.58  4966.2 1521.08    4991 1521.58  5027.5 1524.04  5077.4 1522.98
  5105.7 1526.87  5354.5 1544.16  5423.8 1549.83  5537.2 1565.55  5551.3 1568.91
  5586.5 1583.17  5643.2 1601.14  5671.5 1613.75  5777.5 1646.54  5820.1 1656.05
  5855.7 1660.46  5862.6 1663.84  5898.3 1672.75  5919.3  1680.3  5954.7  1684.8
#Mann= 8 ,-1 , 0
  4525.1     .12       0  4583.2     .07       0  4732.1     .12       0
  4792.7     .07       0  4897.5     .12       0  4965.7     .05       0
    4991     .12       0  5354.5     .07       0
Bank Sta=4965.7,4991
XS Rating Curve= 0 ,0
Exp/Cntr=0.3,0.1

Type RM Length L Ch R = 1 ,42502   ,561,561,561
BEGIN DESCRIPTION:
BLOCK CREEK 74.0
END DESCRIPTION:
XS GIS Cut Line= 3
      2020224.99     13936674.95        2020175.       13936275.
      2019375.04     13935825.02
#Sta/Elev= 30
  4593.2 1556.96  4633.1 1556.96  4666.2 1555.79  4772.2  1546.4  4824.7 1542.44
  4845.1 1539.73  4872.8 1541.63  4953.4 1539.64  4958.5 1534.94  4976.1 1531.65
  4997.3 1515.52  4997.8 1515.02  5022.6 1515.52  5063.5 1522.86  5085.2 1522.46
  5122.5 1515.64  5166.1 1527.08  5230.9 1526.52  5263.1 1527.05    5328 1533.84
  5452.3 1537.18    5555 1546.59  5569.9 1549.14  5614.2 1568.42  5627.3 1576.81
  5710.7 1590.15  5742.1    1597  5781.9 1602.51  5787.9  1607.3  5914.1 1624.72
#Mann= 11 ,-1 , 0
  4593.2     .07       0  4633.1     .12       0  4666.2     .07       0
  4772.2     .12       0  4824.7     .07       0  4997.3     .05       0
  5022.6     .07       0  5230.9     .12       0  5263.1     .07       0
  5710.7    .035       0  5742.1     .07       0
Bank Sta=4997.3,5022.6
XS Rating Curve= 0 ,0
Exp/Cntr=0.3,0.1

Type RM Length L Ch R = 1 ,41941   ,562,562,562
BEGIN DESCRIPTION:
BLOCK CREEK 73.0
END DESCRIPTION:
XS GIS Cut Line= 3
      2020474.98     13936074.97        2020225.       13935725.
      2019925.03     13935425.03
#Sta/Elev= 30
  4574.9 1544.08    4578 1544.06  4603.2 1542.57  4632.6 1541.56  4668.3 1542.16
  4740.5 1539.09    4769 1539.38  4804.7 1536.16  4850.4 1535.09  4890.7 1528.19
  4896.8 1529.03    4903 1527.97  4911.6 1529.12  4932.5 1522.86  4947.2 1513.39
  4978.7 1511.27  4979.2 1510.77  5004.2 1511.27    5005 1513.57  5112.6 1522.86
  5181.8 1529.89  5217.1 1539.16  5231.3 1544.78  5245.4 1552.29  5256.1 1555.33
  5287.8 1565.65  5316.1 1578.68  5325.7  1580.4  5372.7  1588.5  5429.2 1594.47
#Mann= 11 ,-1 , 0
  4574.9    .035       0    4578     .07       0  4603.2    .035       0
  4740.5     .07       0  4850.4     .12       0    4903     .07       0
  4978.7     .05       0  5004.2     .07       0  5112.6     .12       0
  5256.1     .07       0  5325.7    .035       0
Bank Sta=4978.7,5004.2
XS Rating Curve= 0 ,0
Exp/Cntr=0.3,0.1

Type RM Length L Ch R = 1 ,41379   ,565,565,565
BEGIN DESCRIPTION:
BLOCK CREEK 72.0
END DESCRIPTION:
XS GIS Cut Line= 3
        2020675.     13935724.99        2020575.       13935325.
      2020175.01       13935225.
#Sta/Elev= 30
  4587.7 1536.77  4639.2 1535.66  4659.8 1533.58  4693.3 1534.83  4741.7 1533.34
    4817 1533.54  4876.3 1530.83  4902.7 1526.55  4917.5 1523.08  4935.6  1516.5
  4948.5 1515.79  4969.1 1510.73  4969.2 1507.08  4969.7 1506.58  4994.7 1507.08
  4997.4 1509.64  5082.5 1511.94  5100.5 1514.69  5146.9 1530.24    5183  1528.6
  5195.8 1533.21  5224.2 1539.33  5237.1  1543.7  5257.7 1546.35  5288.6 1553.74
  5306.7 1560.94  5340.2 1570.55  5360.8 1579.02  5389.1 1583.34  5412.3 1585.21
#Mann= 5 ,-1 , 0
  4587.7    .035       0  4741.7     .12       0  4902.7     .07       0
  4969.2     .05       0  4994.7     .07       0
Bank Sta=4969.2,4994.7
XS Rating Curve= 0 ,0
Exp/Cntr=0.3,0.1

Type RM Length L Ch R = 1 ,40814   ,534,534,534
BEGIN DESCRIPTION:
BLOCK CREEK 71.0
END DESCRIPTION:
XS GIS Cut Line= 3
      2021824.98     13935824.98        2021025.       13935025.
      2020425.02     13934375.03
#Sta/Elev= 30
  3873.7 1593.11  3916.1 1588.19  3986.8 1565.04  4094.5 1545.59  4128.2 1540.89
  4341.5 1533.91    4725 1528.14  4807.1 1527.64  4866.3 1520.36  4934.3 1513.18
  4962.6 1508.15  4978.1 1502.17  4978.6 1501.67  5003.7 1502.17    5005  1505.4
  5048.3 1515.61  5057.2 1518.89  5089.8 1526.82  5182.8 1529.14    5195 1530.31
  5323.4 1536.47  5343.7 1537.23  5480.4 1545.19  5549.7 1552.95  5613.8 1570.79
  5634.7 1581.53  5677.3 1591.25  5790.7 1605.43  5861.6 1621.75  5889.6 1624.43
#Mann= 14 ,-1 , 0
  3873.7     .07       0  4094.5    .035       0  4341.5     .12       0
    4725    .035       0  4866.3     .12       0  4978.1     .05       0
  5003.7     .12       0  5048.3     .07       0  5057.2     .12       0
  5182.8     .07       0    5195    .035       0  5323.4     .07       0
  5343.7    .035       0  5480.4     .07       0
Bank Sta=4978.1,5003.7
XS Rating Curve= 0 ,0
Exp/Cntr=0.3,0.1

Type RM Length L Ch R = 1 ,40280   ,548,548,548
BEGIN DESCRIPTION:
BLOCK CREEK 70.0
END DESCRIPTION:
XS GIS Cut Line= 3
      2022224.97     13935524.97        2021475.       13934775.
      2020675.03     13934225.02
#Sta/Elev= 30
  3944.5 1592.13  3986.9 1589.46  4028.4 1579.27    4100 1554.76  4164.5 1542.37
    4298 1532.58    4462 1529.45  4764.7 1524.93  4863.7 1526.03  4934.4 1514.86
  4962.7 1506.21  4976.8 1505.11  4978.1 1500.02  4978.6 1499.52  5003.8 1500.02
  5033.5 1506.27  5054.5    1507  5063.8 1511.14  5090.3 1519.94  5120.1 1524.19
  5248.6 1526.21  5272.1 1529.96  5319.3 1526.55  5609.9 1532.21  5738.5 1541.96
  5780.1 1549.86  5810.2 1559.35  5875.8 1590.51  5895.2 1592.75  5975.9 1605.46
#Mann= 10 ,-1 , 0
  3944.5     .07       0  4028.4     .12       0  4164.5     .07       0
    4462     .12       0  4978.1     .05       0  5003.8     .12       0
  5063.8     .07       0  5319.3    .035       0  5780.1     .07       0
  5895.2    .035       0
Bank Sta=4978.1,5003.8
XS Rating Curve= 0 ,0
Exp/Cntr=0.3,0.1

Type RM Length L Ch R = 1 ,39732   ,557,557,557
BEGIN DESCRIPTION:
BLOCK CREEK 69.0
END DESCRIPTION:
XS GIS Cut Line= 3
      2021969.04     13934388.33        2021725.       13934375.
      2021118.75     13934330.32
#Sta/Elev= 30
  4755.6  1521.1  4803.1 1521.01  4869.8 1521.42  4920.8 1523.66  4929.9 1524.52
  4939.9 1516.18  4949.9 1504.82  4959.9 1500.13  4967.1 1498.22  4967.6 1497.72
  4992.8 1498.22  4997.5 1499.31  5020.1 1501.15  5030.1 1504.32  5040.1 1505.97
  5066.6 1508.62  5071.6 1508.27  5150.4 1511.92  5190.5 1516.03  5199.8 1517.69
  5212.9 1517.39  5260.7 1520.13  5280.8 1522.71  5290.8 1523.22  5331.5 1522.96
  5391.1 1524.46  5531.4 1525.61  5561.5 1527.18  5581.6 1526.65  5607.9 1527.39
#Mann= 7 ,-1 , 0
  4755.6    .035       0  4803.1     .07       0  4920.8     .12       0
  4967.1     .05       0  4992.8     .12       0  5212.9     .07       0
  5331.5    .035       0
Bank Sta=4967.1,4992.8
XS Rating Curve= 0 ,0
Exp/Cntr=0.3,0.1

Type RM Length L Ch R = 1 ,39175   ,582,582,582
BEGIN DESCRIPTION:
BLOCK CREEK 68.0
END DESCRIPTION:
XS GIS Cut Line= 3
      2021975.01     13933374.98        2021625.       13933875.
      2020825.01       13933925.
#Sta/Elev= 30
  4390.2 1527.64  4426.8 1527.12  4504.9 1513.34  4571.7 1511.69  4683.6 1508.64
  4719.8 1499.68  4763.8 1497.12  4771.9 1494.44  4772.4 1493.94  4797.7 1494.44
  4799.6 1498.74  4805.7 1501.94  4829.2 1509.19  4850.2  1508.4  4856.3 1503.14
  4951.3 1498.27  4978.3 1495.71  4997.5 1498.52  5070.4 1503.69  5212.4 1516.81
  5295.5 1518.94  5327.2 1520.85  5391.3 1526.21  5461.5 1525.84  5541.6 1531.43
  5559.1 1537.26  5651.8 1551.37  5711.5 1581.74    5742  1592.7  5802.1 1598.24
#Mann= 11 ,-1 , 0
  4390.2    .035       0  4571.7     .07       0  4771.9     .05       0
  4797.7     .07       0  4951.3    .035       0  4997.5     .12       0
  5070.4    .035       0  5212.4     .07       0  5295.5    .035       0
  5327.2     .07       0  5711.5    .035       0
Bank Sta=4951.3,4997.5
XS Rating Curve= 0 ,0
Exp/Cntr=0.3,0.1

Type RM Length L Ch R = 1 ,38593   ,581,581,581
BEGIN DESCRIPTION:
BLOCK CREEK 67.0
END DESCRIPTION:
XS GIS Cut Line= 3
      2021925.01       13933325.        2021525.       13933325.
      2020874.99       13933175.
#Sta/Elev= 30
  4599.6 1528.42  4629.6 1525.43  4658.1  1514.8  4679.6 1508.69  4769.6 1507.42
  4849.6 1499.88  4889.6 1499.43  4936.8 1493.58  4959.6 1492.13  4969.6 1493.54
  4973.2 1490.69  4973.8 1490.19    5006 1490.69  5018.4 1505.42  5023.6 1505.04
  5030.4  1511.5  5050.9 1513.73  5290.4 1520.64  5389.6 1526.77  5430.6 1536.13
  5461.4  1539.6  5509.3 1551.29  5543.5 1557.12  5552.1  1561.3  5574.3 1567.98
  5584.6  1574.1  5605.1 1577.64  5635.9 1585.53  5642.7 1589.41  5666.7 1592.42
#Mann= 5 ,-1 , 0
  4599.6    .035       0  4658.1     .07       0  4936.8    .035       0
  4973.2    .035       0    5006    .035       0
Bank Sta=4973.2,5006
XS Rating Curve= 0 ,0
Exp/Cntr=0.3,0.1

Type RM Length L Ch R = 1 ,38012   ,1103,1103,1103
BEGIN DESCRIPTION:
BLOCK CREEK 66.0
END DESCRIPTION:
XS GIS Cut Line= 3
      2022202.38     13933223.52        2021625.       13932775.
      2021024.97     13932574.99
#Sta/Elev= 30
  4269.4 1522.18  4468.6 1519.75  4530.8 1519.67  4586.9  1510.2  4658.6 1502.88
  4686.5 1502.47  4694.6 1505.39  4705.3 1505.27  4803.9 1502.03  4872.9 1495.99
    4933 1496.37  4972.5 1492.71  5003.2  1493.7  5005.2 1487.35  5005.7 1486.85
    5038 1487.35  5053.7  1488.6  5074.3 1496.78  5095.4  1499.5  5116.5 1506.06
  5148.1 1510.48  5323.6 1514.91    5380 1517.57  5422.1 1522.12  5474.9 1537.92
  5538.1 1549.49  5559.2 1558.69  5590.8 1578.41  5611.9  1584.4    5633 1584.79
#Mann= 10 ,-1 , 0
  4269.4     .12       0  4468.6    .035       0  4705.3     .07       0
  4803.9     .12       0    4933     .07       0  5005.2     .05       0
    5038     .07       0  5053.7    .035       0  5323.6     .07       0
  5422.1    .035       0
Bank Sta=5005.2,5038
XS Rating Curve= 0 ,0
Exp/Cntr=0.3,0.1

Type RM Length L Ch R = 1 ,37462   ,552,552,552
BEGIN DESCRIPTION:
BLOCK CREEK 65.0
END DESCRIPTION:
XS GIS Cut Line= 3
      2022024.96     13932125.01        2021575.       13932275.
      2021124.97       13932325.
#Sta/Elev= 30
  4531.4 1511.27  4594.6 1511.71  4615.2 1506.49  4636.8 1508.07  4657.8 1507.66
  4710.6 1499.26    4816 1495.31  4858.1  1490.6  4931.9 1491.89  4942.5 1490.85
  4957.4 1486.07    4958 1485.57  4990.8 1486.07  5003.1 1489.17  5017.6  1490.5
    5056 1497.21  5076.1 1506.25  5136.5 1510.38    5217 1512.65  5247.2  1517.8
  5263.3  1523.1  5297.5 1534.13  5347.8 1541.44  5367.9 1546.79    5378 1550.17
  5398.1 1560.16  5408.2 1563.29  5418.2 1564.91  5431.8 1564.36  5458.5 1564.75
#Mann= 7 ,-1 , 0
  4531.4    .035       0  4615.2     .07       0  4957.4     .05       0
  4990.8     .07       0  5017.6    .035       0  5263.3     .07       0
  5431.8    .035       0
Bank Sta=4957.4,4990.8
XS Rating Curve= 0 ,0
Exp/Cntr=0.3,0.1

Type RM Length L Ch R = 1 ,36910   ,576,576,576
BEGIN DESCRIPTION:
BLOCK CREEK 64.0
END DESCRIPTION:
XS GIS Cut Line= 3
      2022075.04     13931925.01        2021675.       13931775.
      2021075.01       13931875.
#Sta/Elev= 30
  4576.6 1511.72  4673.4 1508.81    4737 1507.11  4800.9 1507.99  4817.8 1505.49
  4848.1 1505.54    4873  1498.8  4878.3 1499.48  4903.3  1493.2  4933.5 1490.92
  4977.3 1483.38  4977.9 1482.88  5010.8 1483.38  5031.7  1489.1  5064.7 1489.21
  5145.8 1492.93  5158.4    1494  5176.2 1497.85  5257.3  1501.7  5280.1 1504.26
  5282.6 1506.19    5308 1514.92  5358.7 1521.27  5409.4 1532.55  5490.5 1541.88
  5513.2 1545.59  5523.4 1547.93  5541.1 1555.24  5561.4 1560.08  5612.1 1564.27
#Mann= 6 ,-1 , 0
  4576.6     .07       0  4673.4    .035       0    4737     .07       0
  4977.3    .035       0  5010.8     .07       0  5513.2     .07       0
Bank Sta=4977.3,5010.8
XS Rating Curve= 0 ,0
Exp/Cntr=0.3,0.1

Type RM Length L Ch R = 1 ,36334   ,567,567,567
BEGIN DESCRIPTION:
BLOCK CREEK 63.0
END DESCRIPTION:
XS GIS Cut Line= 3
      2022175.03     13931525.02        2021825.       13931325.
        2021025.       13931575.
#Sta/Elev= 30
  4606.8 1506.13  4723.5 1504.72  4797.6 1504.93  4848.7 1502.87  4899.8 1504.02
  4906.3 1502.87  4915.7 1494.19  4921.1 1495.36  4929.3 1480.39  4970.2 1478.66
  4970.8 1478.16  5003.7 1478.66  5007.1 1486.98  5031.2 1487.38  5041.4 1489.24
  5083.3 1488.23  5135.7 1490.97    5209 1487.61  5387.1  1493.3  5464.1 1498.04
  5554.7 1513.16  5561.6 1516.08  5566.8 1513.94  5571.5 1514.91  5617.6 1521.78
  5631.8 1526.18  5638.6 1530.99  5734.4  1541.5  5806.2 1555.72  5848.1 1559.84
#Mann= 7 ,-1 , 0
  4606.8    .035       0  4723.5     .07       0  4921.1     .12       0
  4970.2     .05       0  5003.7     .12       0  5031.2    .035       0
  5571.5     .07       0
Bank Sta=4970.2,5003.7
XS Rating Curve= 0 ,0
Exp/Cntr=0.3,0.1

Type RM Length L Ch R = 1 ,35767   ,550,550,550
BEGIN DESCRIPTION:
BLOCK CREEK 62.0
END DESCRIPTION:
XS GIS Cut Line= 3
      2022337.78     13931084.61        2021725.       13930825.
      2020925.02     13931174.99
#Sta/Elev= 30
  4330.4 1502.68  4575.4 1502.94  4648.4 1500.71  4713.5  1501.2  4787.8 1496.72
    4934 1494.38  4952.2 1486.68  4957.7 1488.15  4963.3 1484.78  4981.4 1481.31
  4986.8 1482.48  4993.2 1478.61  4999.2 1477.98  5000.9 1476.19  5001.6 1475.69
  5034.5 1476.19  5039.6 1484.04  5050.5 1485.53  5126.9 1483.09  5132.7 1485.71
  5179.5 1489.17  5301.5 1487.93    5359 1490.03  5458.6 1494.11  5476.2 1497.49
  5528.8 1513.79  5609.9 1522.38  5680.1 1534.16  5755.7 1542.72  5869.1 1552.32
#Mann= 7 ,-1 , 0
  4330.4    .035       0  4648.4     .07       0  4787.8     .12       0
  4999.2    .035       0  5000.9    .035       0  5034.5    .035       0
    5359     .07       0
Bank Sta=5000.9,5034.5
XS Rating Curve= 0 ,0
Exp/Cntr=0.3,0.1

Type RM Length L Ch R = 1 ,35217   ,547,547,547
BEGIN DESCRIPTION:
BLOCK CREEK 61.0
END DESCRIPTION:
XS GIS Cut Line= 3
        2022375.       13930325.        2021575.       13930325.
      2021124.97       13930375.
#Sta/Elev= 30
    4200 1505.21    4280 1502.48  4344.4  1497.6    4470 1491.47  4541.6 1490.13
    4600  1489.9    4690 1493.76  4738.8 1490.51    4770 1487.28  4837.3 1487.02
    4880 1488.08  4935.9 1482.06    4950 1481.31  4980.7 1474.84  4981.3 1474.34
  5014.3 1474.84  5020.1 1477.14  5040.2 1477.16  5060.4 1483.27  5096.4  1483.1
    5161 1483.23  5181.1 1485.74  5201.2 1491.95  5221.4 1495.96  5241.5 1496.81
  5352.2 1496.89  5382.3 1500.45  5427.1 1513.07  5432.1  1513.7  5452.8 1514.53
#Mann= 12 ,-1 , 0
    4200     .12       0  4344.4    .035       0  4541.6     .12       0
  4738.8     .07       0  4837.3     .12       0  4935.9    .035       0
  4980.7    .035       0  5014.3    .035       0  5096.4     .07       0
  5241.5    .035       0  5427.1     .07       0  5432.1    .035       0
Bank Sta=4980.7,5014.3
XS Rating Curve= 0 ,0
Exp/Cntr=0.3,0.1

Type RM Length L Ch R = 1 ,34670   ,563,563,563
BEGIN DESCRIPTION:
BLOCK CREEK 60.0
END DESCRIPTION:
XS GIS Cut Line= 4
      2022054.16     13929733.44        2021625.       13929825.
      2021323.58     13929907.55      2021037.47     13930276.22
#Sta/Elev= 30
  4561.2 1497.76  4652.4 1493.32  4693.4 1483.57  4737.8 1479.99  4744.4 1478.35
  4754.6 1471.71  4775.1 1475.95  4787.4 1481.21  4867.9 1482.52  4925.7 1479.23
  4975.3 1477.93  4980.4 1478.99  4989.8 1476.38  4993.6 1471.51  4994.2 1471.01
  5027.2 1471.51  5041.5 1473.22  5051.7  1476.2  5056.9 1474.52  5062.2 1478.81
  5072.6 1483.58  5091.4 1489.91  5263.4 1487.98  5416.6 1488.41  5559.6 1492.39
  5651.1 1496.02  5688.1 1498.69  5704.3 1501.75  5729.7  1508.9  5779.2 1513.64
#Mann= 6 ,-1 , 0
  4561.2     .12       0  4867.9     .07       0  4993.6     .05       0
  5027.2     .07       0  5263.4    .035       0  5704.3     .07       0
Bank Sta=4993.6,5027.2
XS Rating Curve= 0 ,0
Exp/Cntr=0.3,0.1

Type RM Length L Ch R = 1 ,34107   ,233,233,233
BEGIN DESCRIPTION:
BLOCK CREEK 59.0
END DESCRIPTION:
XS GIS Cut Line= 3
      2022324.98     13928525.03        2021625.       13929325.
      2021024.99     13930125.02
#Sta/Elev= 30
    3932 1562.75    3960 1559.09  4016.9 1533.55  4052.9 1524.77  4088.1 1517.96
    4109 1511.54  4172.6 1505.13  4194.4 1506.85  4278.9 1500.34    4407 1498.58
  4505.7 1493.61  4698.2 1492.28  4838.3 1492.21  4888.7 1477.61  4923.5 1474.32
    4967 1475.42  4968.9 1469.35  4969.9 1468.85  5006.9 1469.35  5052.3  1471.9
  5073.1 1477.82  5087.3 1479.16    5259 1484.35  5327.5 1485.49  5430.4 1489.34
    5465 1488.81  5601.8 1486.37  5823.1 1488.87  5916.9 1493.07    5995 1499.49
#Mann= 13 ,-1 , 0
    3932     .12       0  4052.9    .035       0  4698.2     .07       0
  4838.3     .12       0  4923.5     .07       0  4968.9     .05       0
  5006.9     .07       0  5087.3     .12       0    5259     .07       0
  5327.5     .12       0  5430.4    .035       0    5465     .07       0
  5601.8    .035       0
Bank Sta=4968.9,5006.9
XS Rating Curve= 0 ,0
Exp/Cntr=0.3,0.1

Type RM Length L Ch R = 1 ,33874   ,1906,1906,1906
BEGIN DESCRIPTION:
BLOCK CREEK 58.0
END DESCRIPTION:
XS GIS Cut Line= 3
      2022262.82     13928499.98      2021427.19     13929224.41
      2020924.99     13930125.02
#Sta/Elev= 30
  3894.4 1562.29    3939 1539.78    3966 1530.03  4045.4 1514.47    4052  1510.3
  4088.2 1502.06  4215.4 1499.47    4315  1493.7  4575.1 1490.61  4799.3 1490.17
    4816  1490.3  4867.9 1489.17  4888.7 1477.41  4896.4 1477.15    4903 1472.98
  4938.1 1473.36  4976.1 1468.24  4977.1 1467.74  5014.1 1468.24  5046.8 1471.47
  5054.3 1475.76  5069.7 1477.34  5302.3 1482.13  5487.5 1481.28    5562 1485.08
  5655.5 1483.25    5796 1486.36  5920.6 1494.28  5991.5 1509.44  6031.5 1510.57
#Mann= 9 ,-1 , 0
  3894.4     .12       0    3966    .035       0  4575.1     .07       0
  4799.3     .12       0    4816     .07       0  4976.1     .05       0
  5014.1     .07       0  5302.3    .035       0  5991.5     .07       0
Bank Sta=4976.1,5014.1
XS Rating Curve= 0 ,0
Exp/Cntr=0.3,0.1

Type RM Length L Ch R = 1 ,31968   ,535,535,535
BEGIN DESCRIPTION:
BLOCK CREEK 57.0
END DESCRIPTION:
XS GIS Cut Line= 3
      2021130.23     13929124.06        2020175.       13929075.
      2019411.09     13928925.42
#Sta/Elev= 30
  4043.1 1482.92  4178.5 1479.43  4253.9 1482.01  4328.7 1482.42  4348.7 1479.62
  4503.1 1473.46  4561.3 1474.95  4679.5 1475.44  4759.3  1475.2  4876.6 1470.72
  4909.5 1467.63  4949.5 1468.53  4969.5 1459.94  4988.8 1456.94  4989.8 1456.44
  5030.8 1456.94  5040.3 1465.64  5074.6 1484.29  5111.7 1509.58  5121.9 1512.84
  5274.3 1514.25  5385.8 1517.12  5468.3 1524.82  5493.9 1522.91  5536.8 1525.37
  5580.4 1526.76  5620.3 1532.48  5712.9 1540.26  5751.3 1549.51    5778 1551.29
#Mann= 12 ,-1 , 0
  4043.1    .035       0  4253.9     .07       0  4503.1    .035       0
  4561.3     .07       0  4679.5     .12       0  4876.6     .07       0
  4988.8     .05       0  5030.8     .07       0  5074.6     .12       0
  5274.3     .07       0  5536.8    .035       0  5620.3     .07       0
Bank Sta=4988.8,5030.8
XS Rating Curve= 0 ,0
Exp/Cntr=0.3,0.1

Type RM Length L Ch R = 1 ,31433   ,500,500,500
BEGIN DESCRIPTION:
BLOCK CREEK 56.0
END DESCRIPTION:
XS GIS Cut Line= 4
      2021258.86     13929058.78      2021182.68     13929023.73
        2020475.       13928675.      2020208.63     13928486.18
#Sta/Elev= 30
  4132.6 1486.33  4199.4 1484.92  4227.7 1482.34  4325.4 1479.01  4429.9 1479.12
  4469.2  1481.2  4481.4 1478.03    4526 1472.18  4564.6  1469.2  4654.5 1469.91
  4751.1 1466.65  4764.9 1466.72  4804.7 1466.87  4884.7 1463.25  4907.1 1464.37
  4946.5 1463.28    4952 1460.27  4969.4 1458.26  4981.6 1455.41  4982.6 1454.91
  5023.6 1455.41  5027.6 1464.94  5042.2 1476.85  5048.5 1480.27  5054.6 1487.61
  5091.2 1488.34    5181  1494.1    5200 1495.09  5327.8 1502.51  5331.9 1503.91
#Mann= 8 ,-1 , 0
  4132.6    .035       0  4751.1     .07       0  4764.9    .035       0
  4969.4     .07       0  4981.6     .05       0  5023.6     .07       0
    5181    .035       0    5200     .07       0
Bank Sta=4981.6,5023.6
XS Rating Curve= 0 ,0
Exp/Cntr=0.3,0.1

Type RM Length L Ch R = 1 ,30933   ,566,566,566
BEGIN DESCRIPTION:
BLOCK CREEK 55.0
END DESCRIPTION:
XS GIS Cut Line= 4
      2021443.42     13928882.75      2021356.93     13928837.27
        2020925.       13928575.      2020575.04     13928375.02
#Sta/Elev= 30
  4390.7 1486.92  4505.3 1485.68  4526.7 1486.37    4579 1482.66  4621.6 1482.49
  4637.1 1480.77  4676.9 1479.95  4710.7 1479.47  4724.7 1475.94  4747.5 1474.11
  4759.6 1471.91  4768.9 1470.34  4774.7 1470.46  4790.2 1466.81  4805.7 1464.74
  4869.7 1462.37    4891 1463.27    4922 1462.39  4949.2 1458.32  4964.7 1457.02
  4969.8 1455.12  4970.8 1454.62  5011.8 1455.12  5016.8 1459.26  5039.1 1463.13
  5066.4 1473.36  5109.6 1481.03  5122.9 1481.58  5311.5 1483.21  5396.8 1483.32
#Mann= 7 ,-1 , 0
  4390.7    .035       0  4676.9     .07       0  4759.6     .12       0
  4969.8     .05       0  5011.8     .12       0  5122.9     .07       0
  5311.5    .035       0
Bank Sta=4969.8,5011.8
XS Rating Curve= 0 ,0
Exp/Cntr=0.3,0.1

Type RM Length L Ch R = 1 ,30367   ,555,555,555
BEGIN DESCRIPTION:
BLOCK CREEK 54.0
END DESCRIPTION:
XS GIS Cut Line= 3
      2022025.02       13928025.        2021225.       13928275.
      2020083.92     13928365.15
#Sta/Elev= 30
  4161.5 1560.55  4179.5 1554.44    4186 1553.22  4360.6 1517.91  4389.3 1507.38
  4433.9 1496.77  4493.9 1491.71  4702.2  1484.3  4910.9 1478.06  4926.3 1477.52
  4936.8 1471.63  4945.7 1462.12    4951 1463.41  4968.2 1454.44    4976 1446.83
    4977 1446.33    5018 1446.83  5019.7 1454.92  5029.8 1457.59  5079.9 1463.91
  5113.5 1464.26  5213.5 1469.56  5240.4 1469.22  5283.9 1475.44  5311.8 1475.62
  5703.3 1484.39  5922.5 1494.71  6022.8 1502.17  6078.5 1510.41  6144.3 1513.23
#Mann= 14 ,-1 , 0
  4161.5    .035       0  4179.5     .07       0    4186    .035       0
  4389.3     .07       0  4493.9    .035       0  4702.2     .12       0
  4910.9     .07       0    4976     .05       0    5018     .07       0
  5113.5     .07       0  5213.5    .035       0  5283.9     .07       0
  5311.8    .035       0  5703.3     .07       0
Bank Sta=4976,5018
XS Rating Curve= 0 ,0
Exp/Cntr=0.3,0.1

Type RM Length L Ch R = 1 ,29812   ,563,563,563
BEGIN DESCRIPTION:
BLOCK CREEK 53.0
END DESCRIPTION:
XS GIS Cut Line= 3
      2021725.01     13927474.99        2021325.       13927775.
      2019912.47     13928312.35
#Sta/Elev= 30
  4491.1 1544.59  4494.6 1544.54  4532.8 1539.18  4548.4 1531.77  4577.6 1524.29
    4632 1516.32  4669.2 1509.05  4741.1 1487.33  4804.7 1483.42  4841.1 1484.98
  4854.7 1481.04  4919.2 1480.64  4969.2 1476.07  4983.8 1466.95    4988  1455.4
  4991.1  1455.4  4991.5 1446.57  4992.5 1446.07  5033.6 1446.57    5061 1457.89
  5144.7 1461.97  5355.4 1467.73  5395.6 1471.75  5540.8 1472.85  5897.4 1483.43
  6130.4    1496  6185.2  1505.5  6221.5 1508.15  6439.7  1515.6  6502.4  1517.5
#Mann= 9 ,-1 , 0
  4491.1     .07       0  4494.6    .035       0    4632     .12       0
  4991.5     .05       0  5033.6     .12       0  5144.7     .07       0
  5355.4    .035       0  5897.4     .07       0  6439.7     .12       0
Bank Sta=4991.5,5033.6
XS Rating Curve= 0 ,0
Exp/Cntr=0.3,0.1

Type RM Length L Ch R = 1 ,29249   ,540,540,540
BEGIN DESCRIPTION:
BLOCK CREEK 52.0
END DESCRIPTION:
XS GIS Cut Line= 3
      2021674.98       13927375.        2021025.       13927325.
      2020224.98     13927975.01
#Sta/Elev= 30
  4348.1 1543.42  4358.1 1542.29  4368.1 1541.58  4388.2 1533.94  4428.3 1524.09
  4488.9 1515.57  4548.7 1506.74  4568.7  1499.6  4598.8 1494.96  4618.9 1486.04
    4649 1486.35  4686.1 1482.48  4883.4 1474.57  4949.9 1468.63  4959.9 1463.06
  4969.9 1446.91  5000.5 1445.91  5001.5 1445.41  5042.6 1445.91  5050.3 1453.61
  5056.7 1454.19  5128.6 1456.84  5184.6 1461.93  5256.5 1463.07  5316.8 1469.96
  5476.7 1469.79  5661.5 1475.45  5852.6 1483.07    5974  1500.5  6030.8 1502.68
#Mann= 9 ,-1 , 0
  4348.1     .07       0  4358.1    .035       0  4488.9     .07       0
  4686.1     .12       0  4883.4     .07       0  5000.5     .05       0
  5042.6     .07       0  5316.8    .035       0  5661.5     .07       0
Bank Sta=5000.5,5042.6
XS Rating Curve= 0 ,0
Exp/Cntr=0.3,0.1
