--- GOSS CREEK.prj (project) ---

Proj Title=GOSS CREEK Base Level Engineering
Current Plan=p01
Default Exp/Contr=0.3,0.1
English Units
Geom File=g01
Flow File=f01
Plan File=p01
BEGIN DESCRIPTION:
GOSS CREEK
END DESCRIPTION:

--- GOSS CREEK.p01 (plan) ---

Plan Title=Multiple Run
Short Identifier=Multiple
Geom File=g01
Flow File=f01
Subcritical Flow
K Sum by GR= 0
Std Step Tol= 0.01
Critical Tol= 0.01
Num of Std Step Trials= 20
Max Error Tol= 0.3
Flow Tol Ratio= 0.001
Split Flow NTrial= 30
Split Flow Tol= 0.02
Split Flow Ratio= 0.02
Log Output Level= 0
Friction Slope Method= 1
Unsteady Friction Slope Method= 2
Unsteady Bridges Friction Slope Method= 1
Parabolic Critical Depth
Global Vel Dist=  1 , 1 , 1
Global Log Level= 0
CheckData=True
Encroach Param= -1, 0, 0, 0
BEGIN DESCRIPTION:
Multiple Run
END DESCRIPTION:

--- GOSS CREEK.f01 (steady flow) ---

Flow Title=Multiple
Number of Profiles=7
Profile Names=10-year,25-year,50-year,1pct_min,100-year,1pct_plu,500-year
River Rch & RM= GOSS CREEK,Reach-1,21895
    2229    3940    5635    3899    7779   15521   14676
River Rch & RM= GOSS CREEK,Reach-1,16423
    2811    5011    7205    5007    9991   19934   19018
River Rch & RM= GOSS CREEK,Reach-1,10991
    2883    5131    7370    5114   10204   20359   19367
River Rch & RM= GOSS CREEK,Reach-1,6929
    3446    6165    8886    6182   12334   24610   23537
Boundary for River Rch & Prof#=GOSS CREEK,Reach-1,1
Up Type=0
Dn Type=3
Dn Slope=0.005
Boundary for River Rch & Prof#=GOSS CREEK,Reach-1,2
Up Type=0
Dn Type=3
Dn Slope=0.005
Boundary for River Rch & Prof#=GOSS CREEK,Reach-1,3
Up Type=0
Dn Type=3
Dn Slope=0.005
Boundary for River Rch & Prof#=GOSS CREEK,Reach-1,4
Up Type=0
Dn Type=3
Dn Slope=0.005
Boundary for River Rch & Prof#=GOSS CREEK,Reach-1,5
Up Type=0
Dn Type=3
Dn Slope=0.005
Boundary for River Rch & Prof#=GOSS CREEK,Reach-1,6
Up Type=0
Dn Type=3
Dn Slope=0.005
Boundary for River Rch & Prof#=GOSS CREEK,Reach-1,7
Up Type=0
Dn Type=3
Dn Slope=0.005

--- GOSS CREEK.g01 (geometry) ---

Geom Title=Existing Conditions

River Reach=GOSS CREEK,Reach-1
Reach XY= 30
      2083775.00     13896075.00      2084621.45     13895323.53
      2084391.41     13894608.20      2084784.80     13894514.52
      2086065.01     13893286.26      2086435.18     13893264.68
      2086573.62     13892915.34      2086374.91     13891902.31
      2086474.33     13891038.91      2086224.91     13890594.87
      2086723.31     13890230.64      2085938.26     13889738.65
      2085821.55     13889126.25      2085524.92     13888856.71
      2085774.32     13888261.08      2085728.45     13887126.25
      2086325.11     13886709.64      2085830.29     13886072.32
      2086277.29     13886069.90      2086881.12     13885426.82
      2087321.30     13885717.32      2087577.70     13885669.64
      2088257.87     13884791.30      2088880.53     13884477.38
      2089569.36     13884376.69      2090023.50     13884821.53
      2090225.07     13884593.29      2089926.62     13884213.17
      2089935.47     13883865.17      2091025.00     13883525.00

Type RM Length L Ch R = 1,21895,472,472,472
BEGIN DESCRIPTION:
GOSS CREEK 47.0
END DESCRIPTION:
XS GIS Cut Line= 3
      2084275.03     13896275.03      2083925.00     13895875.00
      2083875.00     13895574.98
#Sta/Elev= 30
  4468.2 1355.77  4483.5 1355.44  4518.1 1353.07  4538.9 1347.32  4553.2 1345.14
  4588.3 1337.05  4631.0 1331.14  4702.2 1325.96  4843.6 1321.86  4886.3 1318.94
  4935.7 1312.53  4949.9 1311.75  4971.7 1312.58  5002.3 1310.62  5007.8 1309.32
  5008.1 1308.82  5011.9 1309.32  5027.6 1311.62  5032.7 1313.84  5060.6 1316.15
  5080.8 1314.82  5093.5 1316.75  5121.4 1318.17  5131.5 1317.65  5141.7 1315.22
  5202.5 1332.47  5232.9 1343.55  5263.3 1346.46  5283.6 1351.12  5303.9 1352.73
#Mann=4,-1,0
  4468.2   0.035       0  4483.5    0.07       0  5007.8    0.05       0
  5011.9    0.07       0
Bank Sta=5007.8,5011.9
Exp/Cntr=0.3,0.1

Type RM Length L Ch R = 1,21423,430,430,430
BEGIN DESCRIPTION:
GOSS CREEK 46.0
END DESCRIPTION:
XS GIS Cut Line= 3
      2084625.04     13895675.01      2084225.00     13895525.00
      2084025.00     13895475.00
#Sta/Elev= 30
  4578.8 1333.88  4584.8 1333.41  4654.5 1327.45  4664.3 1325.78  4694.2 1317.28
  4739.9 1305.46  4813.8 1304.01  4823.3 1301.36  4823.5 1300.86  4827.5 1301.36
  4835.2 1304.70  4845.0 1305.78  4880.6 1304.03  4905.5 1304.86  4910.8 1303.16
  4930.4 1302.36  4974.0 1305.34  4990.9 1304.57  4996.3 1301.59  5024.1 1304.61
  5029.2 1307.05  5057.6 1312.56  5065.3 1315.15  5070.5 1319.97  5111.7 1329.70
  5140.0 1338.93  5160.7 1347.63  5181.3 1350.75  5201.9 1356.34  5212.2 1356.70
#Mann=5,-1,0
  4578.8    0.07       0  4584.8   0.035       0  4694.2    0.07       0
  4823.3    0.05       0  4827.5    0.07       0
Bank Sta=4823.3,4827.5
Exp/Cntr=0.3,0.1

Type RM Length L Ch R = 1,20993,459,459,459
BEGIN DESCRIPTION:
GOSS CREEK 45.0
END DESCRIPTION:
XS GIS Cut Line= 3
      2084675.03     13895425.01      2084575.00     13895375.00
      2084425.04     13895325.01
#Sta/Elev= 30
  4888.2 1331.51  4891.0 1331.51  4896.6 1329.95  4902.2 1329.52  4910.6 1328.55
  4924.6 1325.32  4933.0 1322.43  4941.3 1318.88  4955.3 1313.82  4963.7 1309.53
  4969.3 1305.69  4977.7 1300.32  4991.6 1296.24  4997.2 1295.62  5003.5 1295.61
  5008.3 1295.53  5008.7 1295.03  5012.5 1295.03  5012.8 1295.53  5021.1 1298.55
  5029.7 1299.77  5031.7 1300.05  5042.2 1299.84  5063.3 1301.40  5073.8 1304.75
  5084.4 1308.66  5105.4 1309.20  5116.0 1310.14  5126.5 1310.76  5158.1 1311.54
#Mann=5,-1,0
  4888.2    0.07       0  5003.5   0.035       0  5008.3    0.05       0
  5012.8   0.035       0  5029.7    0.07       0
Bank Sta=5008.3,5012.8
Exp/Cntr=0.3,0.1

Type RM Length L Ch R = 1,20534,467,467,467
BEGIN DESCRIPTION:
GOSS CREEK 44.0
END DESCRIPTION:
XS GIS Cut Line= 3
      2084923.36     13895182.80      2084525.00     13894975.00
      2084174.99     13894825.00
#Sta/Elev= 30
  4544.1 1344.97  4576.8 1338.33  4698.0 1328.60  4792.0 1324.18  4830.6 1316.18
  4884.5 1312.15  4903.2 1311.06  4913.3 1306.69  4918.9 1307.75  4957.9 1295.39
  4963.1 1297.40  4979.5 1291.52  4985.2 1292.74  5012.9 1287.38  5013.2 1286.88
  5017.4 1287.38  5036.9 1287.68  5055.1 1291.51  5136.7 1291.61  5154.8 1294.93
  5160.2 1293.18  5189.2 1300.18  5207.4 1308.64  5212.8 1307.96  5230.9 1314.54
  5236.4 1313.56  5254.5 1320.71  5312.5 1333.60  5341.6 1348.32  5374.2 1354.18
#Mann=5,-1,0
  4544.1    0.07       0  4884.5   0.035       0  4957.9    0.07       0
  5012.9    0.05       0  5017.4    0.07       0
Bank Sta=5012.9,5017.4
Exp/Cntr=0.3,0.1

Type RM Length L Ch R = 1,20067,438,438,438
BEGIN DESCRIPTION:
GOSS CREEK 43.0
END DESCRIPTION:
XS GIS Cut Line= 3
      2084825.01     13894975.01      2084425.00     13894575.00
      2084225.00     13894575.00
#Sta/Elev= 30
  4433.6 1326.62  4447.8 1325.94  4504.3 1316.99  4590.3 1311.18  4617.5 1307.47
  4659.9 1305.72  4684.3 1303.88  4730.6 1299.49  4787.2 1297.28  4829.6 1293.13
  4843.7 1290.84  4872.0 1289.95  4928.6 1291.19  4985.2 1288.27  4995.8 1286.73
  5001.8 1286.73  5009.3 1284.03  5027.1 1282.88  5027.4 1282.38  5031.6 1282.88
  5049.3 1285.86  5069.3 1285.91  5079.3 1289.60  5089.3 1294.66  5099.3 1303.69
  5139.3 1325.09  5149.3 1332.35  5169.3 1343.44  5189.3 1352.11  5199.3 1353.15
#Mann=5,-1,0
  4433.6    0.07       0  4590.3   0.035       0  4684.3    0.07       0
  5027.1    0.05       0  5031.6    0.07       0
Bank Sta=5027.1,5031.6
Exp/Cntr=0.3,0.1

Type RM Length L Ch R = 1,19629,469,469,469
BEGIN DESCRIPTION:
GOSS CREEK 42.0
END DESCRIPTION:
XS GIS Cut Line= 3
      2084874.98     13894574.97      2084825.00     13894475.00
      2084475.03     13894175.03
#Sta/Elev= 30
  4888.5 1299.61  4889.5 1299.61  4941.6 1296.96  4977.9 1283.54  4995.1 1273.01
  4995.5 1272.51  4999.8 1273.01  5007.4 1273.79  5014.0 1276.95  5028.3 1281.33
  5085.3 1284.16  5113.9 1289.50  5120.4 1292.21  5134.7 1294.96  5156.7 1296.21
  5170.9 1299.34  5177.5 1302.16  5191.8 1303.84  5198.4 1305.70  5248.9 1311.28
  5269.7 1316.78  5290.6 1319.90  5326.8 1323.31  5333.4 1325.69  5347.6 1328.17
  5369.0 1328.72  5382.8 1330.51  5404.7 1335.36  5425.6 1342.29  5461.2 1344.77
#Mann=4,-1,0
  4888.5   0.035       0  4889.5    0.07       0  4995.1    0.05       0
  4999.8    0.07       0
Bank Sta=4995.1,4999.8
Exp/Cntr=0.3,0.1

Type RM Length L Ch R = 1,19160,470,470,470
BEGIN DESCRIPTION:
GOSS CREEK 41.0
END DESCRIPTION:
XS GIS Cut Line= 3
      2085275.02     13894275.02      2085175.00     13894175.00
      2084975.00     13893875.01
#Sta/Elev= 30
  4854.1 1315.11  4882.4 1310.67  4896.6 1306.82  4910.7 1301.61  4924.8 1298.30
  4953.1 1286.39  4960.2 1285.20  4967.3 1281.92  4981.4 1277.72  4992.0 1273.16
  4998.6 1273.16  5003.1 1268.87  5006.7 1268.59  5007.0 1268.09  5011.5 1268.59
  5024.1 1275.48  5045.1 1276.66  5096.2 1277.16  5103.7 1286.10  5111.2 1288.10
  5139.8 1290.63  5168.3 1294.79  5198.4 1296.30  5211.9 1298.93  5219.4 1301.78
  5234.4 1302.67  5255.5 1307.52  5297.5 1311.93  5327.6 1318.75  5356.1 1320.84
#Mann=3,-1,0
  4854.1    0.07       0  5006.7    0.05       0  5011.5    0.07       0
Bank Sta=5006.7,5011.5
Exp/Cntr=0.3,0.1

Type RM Length L Ch R = 1,18690,444,444,444
BEGIN DESCRIPTION:
GOSS CREEK 40.0
END DESCRIPTION:
XS GIS Cut Line= 3
      2085592.12     13894099.66      2085475.00     13893825.00
      2085175.00     13893424.99
#Sta/Elev= 30
  4701.4 1326.71  4762.0 1322.93  4790.3 1316.83  4801.2 1314.83  4856.5 1309.87
  4880.1 1304.97  4891.3 1298.58  4932.8 1290.21  4945.6 1281.87  4956.4 1278.99
  4967.4 1272.20  4985.5 1267.48  4988.5 1265.07  4988.9 1264.57  4993.3 1265.07
  5013.5 1272.44  5057.3 1271.64  5150.0 1277.65  5157.3 1279.20  5178.1 1289.52
  5213.5 1296.40  5236.5 1304.37  5257.3 1309.04  5271.9 1310.22  5300.0 1317.18
  5363.5 1327.79  5392.7 1329.98  5442.7 1341.85  5471.9 1350.98  5500.0 1354.45
#Mann=5,-1,0
  4701.4    0.07       0  4790.3   0.035       0  4801.2    0.07       0
  4988.5    0.05       0  4993.3    0.07       0
Bank Sta=4988.5,4993.3
Exp/Cntr=0.3,0.1

Type RM Length L Ch R = 1,18246,350,350,350
BEGIN DESCRIPTION:
GOSS CREEK 39.0
END DESCRIPTION:
XS GIS Cut Line= 3
      2085775.00     13893925.03      2085775.00     13893525.00
      2085425.01     13893175.01
#Sta/Elev= 30
  4600.3 1295.42  4680.3 1286.84  4720.3 1283.89  4740.3 1279.64  4760.3 1277.04
  4810.3 1273.05  4970.3 1269.88  4995.4 1265.27  4995.7 1264.77  5000.3 1265.27
  5005.9 1265.28  5008.0 1265.29  5014.5 1265.34  5028.6 1268.61  5042.8 1270.06
  5099.3 1267.57  5140.7 1269.79  5151.6 1270.45  5184.2 1273.28  5198.3 1278.03
  5254.9 1303.74  5275.9 1308.96  5288.4 1312.83  5297.3 1315.91  5325.6 1321.44
  5382.2 1330.17  5410.5 1338.58  5459.1 1349.74  5481.2 1353.31  5495.3 1353.71
#Mann=10,-1,0
  4600.3   0.035       0  4995.4   0.035       0  5000.3   0.035       0
  5005.9    0.07       0  5008.0   0.035       0  5140.7    0.07       0
  5151.6   0.035       0  5275.9    0.07       0  5288.4   0.035       0
  5459.1    0.07       0
Bank Sta=4995.4,5000.3
Exp/Cntr=0.3,0.1

Type RM Length L Ch R = 1,17896,537,537,537
BEGIN DESCRIPTION:
GOSS CREEK 38.0
END DESCRIPTION:
XS GIS Cut Line= 3
      2086524.97     13893674.98      2086043.50     13893314.91
      2085939.66     13893103.78
#Sta/Elev= 30
  4392.0 1324.79  4420.1 1322.36  4455.5 1314.55  4499.3 1309.31  4563.9 1288.23
  4570.2 1281.57  4578.5 1279.90  4584.7 1276.08  4605.6 1270.03  4622.1 1267.25
  4678.5 1263.16  4793.4 1264.78  4817.8 1259.82  4818.2 1259.32  4822.7 1259.82
  4841.5 1263.29  4920.1 1263.36  4934.9 1262.91  4964.1 1265.39  4999.9 1260.08
  5060.0 1264.46  5067.3 1269.37  5072.9 1269.02  5082.3 1277.43  5089.8 1287.69
  5095.4 1286.22  5104.6 1291.65  5134.8 1294.61  5171.4 1301.52  5228.5 1305.49
#Mann=6,-1,0
  4392.0   0.035       0  4622.1    0.07       0  4793.4   0.035       0
  4817.8    0.05       0  4822.7   0.035       0  4920.1    0.07       0
Bank Sta=4817.8,4822.7
Exp/Cntr=0.3,0.1

Type RM Length L Ch R = 1,17359,482,482,482
BEGIN DESCRIPTION:
GOSS CREEK 37.0
END DESCRIPTION:
XS GIS Cut Line= 3
      2086706.69     13893373.94      2086475.00     13893175.00
      2086074.99     13893075.00
#Sta/Elev= 30
  4694.7 1306.17  4730.7 1305.73  4750.9 1302.67  4808.2 1297.93  4877.4 1289.38
  4900.8 1286.11  4915.0 1279.69  4935.9 1275.26  4943.6 1269.20  4964.4 1263.58
  4972.1 1257.11  4978.7 1256.75  4986.4 1252.35  4992.9 1251.28  4994.0 1246.81
  4994.4 1246.31  4999.6 1246.81  5003.2 1246.91  5010.4 1248.40  5018.1 1252.85
  5023.3 1252.75  5031.0 1256.22  5041.3 1258.04  5127.9 1260.08  5204.8 1261.43
  5302.0 1264.98  5340.2 1268.49  5353.1 1270.63  5371.2 1276.91  5412.4 1281.75
#Mann=9,-1,0
  4694.7    0.07       0  4750.9    0.12       0  4877.4    0.07       0
  4994.0    0.05       0  4999.6    0.07       0  5003.2   0.035       0
  5127.9    0.07       0  5204.8   0.035       0  5302.0    0.07       0
Bank Sta=4994,4999.6
Exp/Cntr=0.3,0.1

Type RM Length L Ch R = 1,16877,454,454,454
BEGIN DESCRIPTION:
GOSS CREEK 36.0
END DESCRIPTION:
XS GIS Cut Line= 3
      2086975.00     13892675.00      2086575.00     13892725.00
      2086175.03     13892924.99
#Sta/Elev= 30
  4596.9 1304.13  4617.1 1302.06  4634.7 1296.49  4639.7 1296.80  4682.8 1284.25
  4788.4 1269.91  4808.5 1265.33  4848.8 1259.78  4876.6 1257.37  4899.2 1252.59
  4929.5 1248.70  4957.2 1253.29  4994.7 1247.24  4995.1 1246.74  5000.3 1247.24
  5009.2 1248.23  5014.0 1247.77  5022.4 1250.05  5058.7 1251.07  5068.3 1252.81
  5101.2 1253.33  5120.2 1252.39  5187.3 1255.00  5192.9 1254.21  5237.6 1255.50
  5327.0 1259.10  5370.6 1262.04  5416.5 1265.22  5424.9 1267.11  5447.2 1267.95
#Mann=8,-1,0
  4596.9    0.12       0  4682.8    0.07       0  4994.7    0.05       0
  5000.3    0.07       0  5009.2   0.035       0  5068.3    0.07       0
  5101.2   0.035       0  5370.6    0.07       0
Bank Sta=4994.7,5000.3
Exp/Cntr=0.3,0.1

Type RM Length L Ch R = 1,16423,441,441,441
BEGIN DESCRIPTION:
GOSS CREEK 35.0
END DESCRIPTION:
XS GIS Cut Line= 3
      2086624.97     13892275.01      2086525.00     13892325.00
      2086124.99     13892124.99
#Sta/Elev= 30
  4881.7 1262.54  4918.0 1260.07  4985.1 1252.34  4990.7 1248.20  4996.3 1248.20
  5001.9 1245.22  5007.4 1246.77  5015.8 1243.10  5026.6 1242.56  5027.1 1242.06
  5033.0 1242.56  5046.6 1245.81  5052.2 1244.88  5062.8 1246.38  5082.9 1247.71
  5141.6 1248.46  5158.4 1250.77  5172.4 1248.90  5203.1 1249.74  5217.1 1248.74
  5225.5 1250.28  5240.0 1250.52  5320.5 1252.66  5337.3 1255.94  5342.9 1255.84
  5359.6 1259.73  5365.2 1259.77  5382.0 1264.88  5409.9 1269.58  5440.7 1277.16
#Mann=5,-1,0
  4881.7    0.07       0  5026.6    0.05       0  5033.0    0.07       0
  5062.8   0.035       0  5240.0    0.07       0
Bank Sta=5026.6,5033
Exp/Cntr=0.3,0.1

Type RM Length L Ch R = 1,15982,469,469,469
BEGIN DESCRIPTION:
GOSS CREEK 34.0
END DESCRIPTION:
XS GIS Cut Line= 3
      2086775.02     13892075.01      2086375.00     13891925.00
      2086074.96     13891874.99
#Sta/Elev= 30
  4578.8 1269.57  4618.9 1265.07  4654.5 1263.36  4707.8 1259.18  4820.0 1249.94
  4884.1 1246.97  4920.6 1245.10  4941.9 1244.99  4966.0 1242.42  4970.8 1239.18
  4971.3 1238.68  4977.2 1239.18  4990.9 1243.70  5056.7 1245.79  5099.8 1248.52
  5127.7 1255.27  5155.6 1266.07  5160.6 1266.18  5168.2 1269.66  5200.9 1281.39
  5208.8 1284.43  5216.4 1289.77  5221.4 1290.44  5229.1 1294.77  5239.2 1298.99
  5259.5 1305.07  5277.2 1309.06  5289.9 1310.67  5304.5 1311.23  5310.2 1311.35
#Mann=7,-1,0
  4578.8    0.07       0  4707.8   0.035       0  4884.1    0.07       0
  4970.8    0.05       0  4977.2    0.07       0  5200.9   0.035       0
  5304.5    0.07       0
Bank Sta=4970.8,4977.2
Exp/Cntr=0.3,0.1

Type RM Length L Ch R = 1,15513,463,463,463
BEGIN DESCRIPTION:
GOSS CREEK 33.0
END DESCRIPTION:
XS GIS Cut Line= 3
      2086824.98     13891275.01      2086425.00     13891475.00
      2086174.96     13891575.02
#Sta/Elev= 30
  4552.8 1311.03  4589.1 1303.50  4605.9 1294.02  4611.5 1293.72  4628.3 1283.34
  4633.8 1282.53  4650.6 1274.52  4656.2 1274.21  4673.0 1266.13  4678.6 1266.35
  4695.3 1257.36  4717.7 1249.44  4723.5 1249.63  4740.1 1245.27  4762.4 1244.38
  4920.6 1242.44  4969.3 1239.96  4988.4 1235.40  4988.9 1234.90  4994.9 1235.40
  4999.3 1236.62  5032.3 1239.54  5039.0 1244.12  5044.4 1239.93  5063.3 1254.15
  5131.3 1266.67  5206.0 1279.58  5224.8 1286.89  5230.2 1286.83  5269.3 1300.09
#Mann=7,-1,0
  4552.8    0.12       0  4723.5   0.035       0  4920.6    0.07       0
  4988.4   0.035       0  4994.9    0.07       0  4999.3   0.035       0
  5131.3    0.07       0
Bank Sta=4988.4,4994.9
Exp/Cntr=0.3,0.1

Type RM Length L Ch R = 1,15050,472,472,472
BEGIN DESCRIPTION:
GOSS CREEK 32.0
END DESCRIPTION:
XS GIS Cut Line= 3
      2086725.01     13891025.00      2086475.00     13891025.00
      2086075.00     13891425.00
#Sta/Elev= 30
  4745.5 1303.57  4755.5 1301.59  4785.5 1292.44  4811.5 1282.06  4865.5 1265.61
  4895.5 1258.48  4915.5 1251.16  4935.5 1241.79  4945.5 1238.62  4955.5 1237.30
  4985.5 1237.64  5006.3 1233.90  5006.8 1233.40  5012.9 1233.90  5037.9 1234.35
  5066.2 1238.11  5094.5 1237.62  5179.4 1240.51  5264.2 1240.24  5292.5 1243.13
  5334.9 1250.47  5363.2 1256.28  5384.4 1262.75  5433.9 1271.97  5448.1 1275.86
  5478.6 1280.28  5504.6 1288.59  5532.9 1294.58  5547.1 1298.74  5561.2 1300.94
#Mann=5,-1,0
  4745.5    0.12       0  4811.5   0.035       0  5006.3   0.035       0
  5012.9   0.035       0  5478.6    0.07       0
Bank Sta=5006.3,5012.9
Exp/Cntr=0.3,0.1

Type RM Length L Ch R = 1,14578,896,896,896
BEGIN DESCRIPTION:
GOSS CREEK 31.0
END DESCRIPTION:
XS GIS Cut Line= 3
      2086624.98     13890874.99      2086225.00     13890675.00
      2086024.99     13890524.99
#Sta/Elev= 30
  4552.6 1266.72  4656.0 1247.07  4723.1 1238.55  4745.4 1236.86  4790.2 1236.00
  4806.9 1233.51  4863.7 1231.99  4888.0 1231.16  4896.4 1229.11  4902.0 1230.31
  4941.8 1227.97  5021.7 1223.80  5027.9 1223.80  5036.2 1227.59  5042.5 1226.71
  5049.8 1227.34  5057.1 1226.48  5060.0 1222.75  5060.5 1222.25  5066.6 1222.75
  5092.5 1224.18  5099.8 1225.55  5107.1 1228.39  5136.2 1244.74  5149.8 1254.17
  5157.1 1263.33  5199.8 1284.25  5213.3 1292.21  5227.9 1297.14  5249.8 1301.43
#Mann=5,-1,0
  4552.6    0.07       0  4863.7   0.035       0  4941.8    0.07       0
  5060.0    0.05       0  5066.6    0.07       0
Bank Sta=5060,5066.6
Exp/Cntr=0.3,0.1

Type RM Length L Ch R = 1,13682,430,430,430
BEGIN DESCRIPTION:
GOSS CREEK 30.0
END DESCRIPTION:
XS GIS Cut Line= 3
      2087357.38     13889880.55      2086625.00     13890125.00
      2086225.00     13890425.00
#Sta/Elev= 30
  4228.2 1335.27  4315.0 1328.33  4378.3 1314.38  4389.2 1308.58  4409.9 1306.51
  4420.9 1300.40  4441.6 1298.81  4478.8 1287.62  4515.7 1271.64  4605.2 1265.06
  4610.5 1261.60  4636.8 1265.69  4642.1 1260.65  4668.4 1263.11  4673.7 1259.47
  4700.0 1259.96  4705.3 1253.27  4731.6 1252.92  4747.3 1244.06  4936.6 1223.82
  4957.9 1220.52  4994.1 1213.80  4994.6 1213.30  5001.2 1213.80  5050.3 1224.19
  5216.0 1225.42  5259.7 1225.42  5343.0 1227.50  5472.1 1257.96  5500.3 1264.70
#Mann=8,-1,0
  4228.2    0.12       0  4936.6    0.07       0  4957.9   0.035       0
  4994.1   0.035       0  5001.2   0.035       0  5216.0    0.07       0
  5259.7   0.035       0  5472.1    0.07       0
Bank Sta=4994.1,5001.2
Exp/Cntr=0.3,0.1

Type RM Length L Ch R = 1,13252,422,422,422
BEGIN DESCRIPTION:
GOSS CREEK 29.0
END DESCRIPTION:
XS GIS Cut Line= 3
      2086474.99     13889725.01      2086275.00     13889925.00
      2085975.03     13890174.98
#Sta/Elev= 30
  4712.6 1280.07  4726.7 1278.30  4783.3 1265.85  4830.2 1251.55  4839.9 1248.06
  4910.6 1231.44  4967.1 1221.85  4991.9 1216.86  4998.7 1216.86  5009.1 1211.97
  5013.3 1211.45  5013.8 1210.95  5020.5 1211.45  5023.4 1212.65  5037.7 1215.01
  5066.4 1217.59  5187.4 1219.39  5201.7 1223.80  5208.3 1224.90  5216.1 1228.44
  5222.6 1234.33  5236.9 1249.84  5243.4 1251.43  5265.5 1264.73  5279.8 1268.77
  5300.7 1272.52  5321.5 1280.50  5335.8 1282.95  5364.2 1291.57  5385.9 1294.17
#Mann=5,-1,0
  4712.6    0.12       0  4830.2   0.035       0  5013.3   0.035       0
  5020.5   0.035       0  5364.2    0.07       0
Bank Sta=5013.3,5020.5
Exp/Cntr=0.3,0.1

Type RM Length L Ch R = 1,12830,461,461,461
BEGIN DESCRIPTION:
GOSS CREEK 28.0
END DESCRIPTION:
XS GIS Cut Line= 3
      2086324.98     13889525.01      2085925.00     13889725.00
      2085831.70     13890214.20
#Sta/Elev= 30
  4556.6 1276.85  4565.0 1273.92  4570.5 1274.26  4587.3 1268.20  4615.3 1263.21
  4660.2 1243.98  4699.1 1228.15  4735.5 1218.26  4928.3 1215.31  4967.4 1210.83
  4995.4 1212.64  5010.4 1210.71  5010.9 1210.21  5017.6 1210.71  5044.5 1215.08
  5075.0 1223.49  5082.0 1228.48  5087.1 1227.89  5115.8 1240.99  5139.2 1244.58
  5207.4 1261.32  5247.3 1267.08  5265.0 1269.29  5300.7 1272.89  5339.7 1281.54
  5370.3 1284.22  5399.9 1291.61  5405.0 1290.50  5457.1 1300.63  5501.8 1302.59
#Mann=6,-1,0
  4556.6    0.12       0  4660.2   0.035       0  5010.4   0.035       0
  5017.6   0.035       0  5247.3    0.12       0  5265.0    0.07       0
Bank Sta=5010.4,5017.6
Exp/Cntr=0.3,0.1

Type RM Length L Ch R = 1,12369,453,453,453
BEGIN DESCRIPTION:
GOSS CREEK 27.0
END DESCRIPTION:
XS GIS Cut Line= 3
      2086024.96     13889175.03      2085825.00     13889325.00
      2085012.25     13889717.69
#Sta/Elev= 30
  4754.3 1279.91  4767.8 1277.20  4782.4 1271.36  4797.0 1263.19  4803.8 1253.99
  4811.5 1244.62  4861.5 1212.67  4867.8 1210.01  4904.3 1211.14  4926.1 1206.69
  4972.0 1203.32  4972.5 1202.82  4980.2 1203.32  4997.0 1203.99  5001.1 1208.41
  5125.8 1217.86  5170.8 1229.22  5204.7 1241.71  5289.5 1266.28  5362.9 1277.91
  5379.9 1283.10  5392.8 1284.60  5457.8 1296.49  5504.0 1303.97  5569.3 1305.86
  5626.2 1308.25  5662.2 1311.78  5752.6 1315.14  5807.5 1322.54  5906.9 1327.80
#Mann=8,-1,0
  4754.3    0.12       0  4803.8   0.035       0  4972.0   0.035       0
  4980.2   0.035       0  5392.8    0.07       0  5457.8   0.035       0
  5569.3    0.07       0  5807.5   0.035       0
Bank Sta=4972,4980.2
Exp/Cntr=0.3,0.1

Type RM Length L Ch R = 1,11916,476,476,476
BEGIN DESCRIPTION:
GOSS CREEK 26.0
END DESCRIPTION:
XS GIS Cut Line= 3
      2086024.96     13889024.99      2085625.00     13888975.00
      2084939.69     13889061.39
#Sta/Elev= 30
  4596.9 1280.63  4639.7 1274.23  4708.3 1254.42  4727.9 1250.25  4808.5 1224.29
  4947.8 1206.63  5005.8 1197.80  5006.3 1197.30  5014.3 1197.80  5029.3 1200.86
  5050.4 1205.04  5141.1 1204.43  5151.2 1207.59  5191.5 1231.66  5211.6 1252.75
  5231.8 1265.26  5262.0 1272.91  5285.2 1274.61  5352.7 1283.28  5393.1 1284.52
  5439.1 1289.99  5444.1 1287.10  5519.4 1294.19  5524.4 1291.35  5594.6 1296.81
  5599.6 1294.82  5604.7 1298.42  5635.0 1303.01  5679.9 1305.79  5690.7 1308.26
#Mann=7,-1,0
  4596.9    0.12       0  4708.3   0.035       0  4947.8    0.07       0
  5005.8    0.05       0  5014.3    0.07       0  5029.3   0.035       0
  5285.2    0.07       0
Bank Sta=5005.8,5014.3
Exp/Cntr=0.3,0.1

Type RM Length L Ch R = 1,11440,449,449,449
BEGIN DESCRIPTION:
GOSS CREEK 25.0
END DESCRIPTION:
XS GIS Cut Line= 3
      2086025.02     13888675.01      2085625.00     13888575.00
      2085475.03     13888575.00
#Sta/Elev= 30
  4591.9 1282.25  4610.0 1277.19  4622.8 1274.89  4633.2 1270.08  4643.5 1266.85
  4651.2 1261.72  4656.3 1260.66  4674.4 1252.10  4698.2 1242.81  4746.5 1221.77
  4774.9 1210.84  4787.8 1207.79  4799.0 1207.31  4899.8 1204.49  4902.5 1204.29
  4952.7 1201.33  4973.3 1195.94  4981.9 1194.92  4982.4 1194.42  4990.5 1194.92
  4993.9 1198.60  5000.6 1199.66  5014.2 1200.87  5024.2 1203.72  5034.2 1212.89
  5074.2 1231.92  5084.2 1238.08  5134.2 1259.27  5146.4 1263.27  5154.2 1265.59
#Mann=9,-1,0
  4591.9    0.12       0  4698.2    0.07       0  4799.0   0.035       0
  4899.8    0.07       0  4902.5    0.12       0  4981.9    0.05       0
  4990.5    0.12       0  5000.6    0.07       0  5146.4   0.035       0
Bank Sta=4981.9,4990.5
Exp/Cntr=0.3,0.1

Type RM Length L Ch R = 1,10991,465,465,465
BEGIN DESCRIPTION:
GOSS CREEK 24.0
END DESCRIPTION:
XS GIS Cut Line= 3
      2086024.96     13888125.01      2085775.00     13888175.00
      2085425.02     13888374.99
#Sta/Elev= 30
  4745.2 1277.52  4775.8 1270.64  4785.9 1263.50  4796.1 1252.91  4862.2 1210.26
  4877.7 1200.56  4887.9 1198.22  4908.3 1196.59  4938.9 1197.98  4969.5 1197.42
  5003.0 1194.76  5009.5 1189.47  5010.0 1188.97  5018.1 1189.47  5023.1 1195.97
  5029.6 1197.04  5072.8 1198.90  5088.6 1201.94  5097.0 1201.96  5131.8 1203.52
  5153.4 1207.49  5161.4 1210.17  5212.5 1217.96  5234.1 1223.31  5250.9 1229.86
  5279.8 1240.97  5361.9 1260.69  5373.7 1262.63  5389.5 1268.35  5403.2 1269.98
#Mann=8,-1,0
  4745.2    0.12       0  4862.2   0.035       0  5009.5   0.035       0
  5018.1   0.035       0  5097.0    0.12       0  5250.9    0.07       0
  5279.8   0.035       0  5361.9    0.07       0
Bank Sta=5009.5,5018.1
Exp/Cntr=0.3,0.1

Type RM Length L Ch R = 1,10526,448,448,448
BEGIN DESCRIPTION:
GOSS CREEK 23.0
END DESCRIPTION:
XS GIS Cut Line= 3
      2085924.97     13887775.00      2085675.00     13887775.00
      2085325.03     13887825.00
#Sta/Elev= 30
  4754.3 1267.87  4756.8 1267.87  4764.3 1265.39  4774.3 1260.67  4844.3 1239.31
  4884.3 1221.21  4898.0 1217.10  4904.3 1215.41  4934.3 1197.83  4944.3 1194.41
  4964.3 1190.25  4969.8 1190.14  4970.3 1189.64  4978.8 1190.14  5001.8 1193.88
  5026.3 1195.01  5105.3 1197.30  5125.5 1200.33  5135.6 1203.19  5155.8 1210.95
  5165.9 1215.58  5176.0 1218.85  5206.3 1232.50  5226.5 1239.56  5256.8 1248.50
  5307.3 1258.85  5327.5 1264.64  5337.6 1266.25  5347.7 1269.95  5357.8 1271.63
#Mann=5,-1,0
  4754.3    0.12       0  4898.0   0.035       0  4969.8   0.035       0
  4978.8   0.035       0  5026.3    0.07       0
Bank Sta=4969.8,4978.8
Exp/Cntr=0.3,0.1

Type RM Length L Ch R = 1,10078,451,451,451
BEGIN DESCRIPTION:
GOSS CREEK 22.0
END DESCRIPTION:
XS GIS Cut Line= 3
      2086025.01     13887625.01      2085675.00     13887325.00
      2085475.00     13887225.00
#Sta/Elev= 30
  4543.4 1272.80  4556.3 1270.38  4579.1 1266.46  4595.3 1260.88  4663.6 1241.13
  4671.3 1236.47  4706.4 1224.07  4820.0 1199.98  4853.8 1195.77  4940.2 1193.95
  4954.4 1190.95  4983.0 1188.74  4992.8 1186.27  4993.3 1185.77  5001.8 1186.27
  5007.2 1186.43  5010.6 1188.60  5017.9 1190.39  5049.1 1191.79  5085.4 1188.85
  5093.8 1191.39  5107.8 1198.94  5116.2 1205.15  5124.6 1215.37  5152.5 1232.69
  5169.3 1261.73  5174.9 1263.54  5191.7 1273.45  5205.6 1277.91  5228.0 1280.94
#Mann=8,-1,0
  4543.4    0.07       0  4556.3    0.12       0  4595.3    0.07       0
  4853.8   0.035       0  4992.8   0.035       0  5001.8   0.035       0
  5010.6    0.07       0  5017.9   0.035       0
Bank Sta=4992.8,5001.8
Exp/Cntr=0.3,0.1

Type RM Length L Ch R = 1,9627,446,446,446
BEGIN DESCRIPTION:
GOSS CREEK 21.0
END DESCRIPTION:
XS GIS Cut Line= 3
      2086325.01     13887325.01      2085925.00     13887025.00
      2085765.74     13886950.34
#Sta/Elev= 30
  4500.0 1277.74  4542.7 1269.87  4563.6 1264.47  4581.3 1256.89  4613.6 1246.42
  4650.0 1230.82  4686.5 1220.58  4707.3 1211.83  4742.7 1203.24  4778.1 1197.68
  4842.7 1191.40  4909.5 1190.55  4950.0 1191.18  4986.5 1187.46  4992.7 1184.30
  5008.7 1183.02  5009.6 1180.39  5010.1 1179.89  5018.7 1180.39  5031.5 1182.37
  5054.3 1189.68  5066.3 1198.42  5077.1 1200.63  5088.4 1209.71  5099.4 1212.60
  5111.0 1222.24  5121.5 1225.13  5133.8 1233.03  5156.6 1241.09  5175.9 1245.58
#Mann=5,-1,0
  4500.0    0.12       0  4581.3    0.07       0  4909.5    0.12       0
  5009.6    0.05       0  5018.7    0.12       0
Bank Sta=5009.6,5018.7
Exp/Cntr=0.3,0.1

Type RM Length L Ch R = 1,9181,445,445,445
BEGIN DESCRIPTION:
GOSS CREEK 20.0
END DESCRIPTION:
XS GIS Cut Line= 3
      2086524.97     13886824.99      2086275.00     13886775.00
      2085679.47     13886856.50
#Sta/Elev= 30
  4745.4 1277.33  4765.8 1274.08  4776.0 1269.69  4816.8 1244.23  4827.0 1234.12
  4837.1 1228.12  4857.5 1212.87  4867.7 1207.92  4898.3 1184.07  4917.1 1182.53
  4949.3 1186.17  4959.5 1185.77  4975.3 1181.41  4975.8 1180.91  4984.5 1181.41
  4999.8 1181.64  5041.5 1182.13  5099.7 1187.20  5141.6 1186.35  5199.6 1190.43
  5323.3 1200.82  5373.8 1207.12  5402.5 1207.22  5407.5 1210.75  5464.6 1214.06
  5505.0 1222.35  5551.9 1236.54  5557.0 1233.63  5575.6 1240.80  5601.4 1246.60
#Mann=7,-1,0
  4745.4    0.12       0  4917.1    0.07       0  4975.3   0.035       0
  4984.5    0.07       0  4999.8   0.035       0  5099.7    0.07       0
  5199.6    0.12       0
Bank Sta=4975.3,4984.5
Exp/Cntr=0.3,0.1

Type RM Length L Ch R = 1,8736,328,328,328
BEGIN DESCRIPTION:
GOSS CREEK 19.0
END DESCRIPTION:
XS GIS Cut Line= 3
      2086375.00     13886475.00      2086075.00     13886475.00
      2085675.00     13886625.00
#Sta/Elev= 30
  4699.5 1256.33  4739.5 1245.63  4789.5 1225.88  4809.5 1220.53  4849.5 1203.31
  4869.5 1197.08  4909.5 1187.74  4934.5 1183.62  4959.5 1178.37  4992.4 1176.08
  4992.9 1175.58  5001.6 1176.08  5002.9 1176.32  5014.6 1180.43  5039.5 1181.39
  5044.9 1183.26  5125.0 1184.49  5149.0 1186.42  5185.5 1193.16  5234.5 1205.49
  5240.7 1209.40  5246.0 1210.36  5265.6 1218.68  5301.2 1228.16  5341.3 1245.21
  5356.4 1247.47  5381.3 1254.50  5405.3 1257.80  5411.6 1261.99  5426.7 1262.47
#Mann=5,-1,0
  4699.5    0.12       0  4934.5   0.035       0  4992.4   0.035       0
  5001.6   0.035       0  5002.9    0.12       0
Bank Sta=4992.4,5001.6
Exp/Cntr=0.3,0.1

Type RM Length L Ch R = 1,8408,686,686,686
BEGIN DESCRIPTION:
GOSS CREEK 18.0
END DESCRIPTION:
XS GIS Cut Line= 3
      2086339.80     13886365.89      2086085.58     13886207.53
      2085558.13     13886307.20
#Sta/Elev= 30
  4485.8 1228.51  4491.4 1228.51  4512.5 1223.64  4539.6 1221.00  4576.2 1208.21
  4597.5 1203.02  4628.7 1198.31  4686.0 1189.81  4780.4 1182.23  4860.7 1181.54
  4909.7 1182.67  4969.1 1178.65  4984.8 1174.69  4985.3 1174.19  4994.1 1174.69
  5020.0 1178.59  5081.0 1178.54  5101.4 1183.69  5111.6 1187.87  5119.2 1194.69
  5131.9 1203.60  5171.6 1229.75  5176.7 1230.71  5193.0 1246.02  5203.2 1251.44
  5217.1 1256.29  5229.0 1261.13  5234.1 1260.94  5254.0 1266.01  5322.1 1271.90
#Mann=6,-1,0
  4485.8    0.12       0  4628.7   0.035       0  4860.7    0.12       0
  4984.8    0.05       0  4994.1    0.12       0  5217.1    0.07       0
Bank Sta=4984.8,4994.1
Exp/Cntr=0.3,0.1

Type RM Length L Ch R = 1,7722,316,316,316
BEGIN DESCRIPTION:
GOSS CREEK 17.0
END DESCRIPTION:
XS GIS Cut Line= 2
      2086414.80     13886336.70      2086077.77     13885779.15
#Sta/Elev= 30
  4694.5 1239.30  4698.4 1239.30  4708.9 1234.17  4731.5 1228.20  4790.0 1220.23
  4820.3 1208.07  4848.4 1200.36  4957.2 1186.49  5000.3 1172.45  5009.6 1170.33
  5015.4 1171.94  5019.0 1168.19  5019.5 1167.69  5028.3 1168.19  5046.5 1171.23
  5052.3 1170.36  5067.8 1174.76  5072.5 1174.35  5140.5 1179.13  5162.9 1186.00
  5198.9 1192.44  5211.4 1196.59  5221.1 1198.20  5242.4 1206.34  5269.6 1218.91
  5300.6 1224.94  5306.5 1227.93  5322.0 1231.53  5327.8 1234.63  5346.0 1239.08
#Mann=5,-1,0
  4694.5    0.12       0  4820.3   0.035       0  5019.0   0.035       0
  5028.3   0.035       0  5072.5    0.12       0
Bank Sta=5019,5028.3
Exp/Cntr=0.3,0.1

Type RM Length L Ch R = 1,7406,477,477,477
BEGIN DESCRIPTION:
GOSS CREEK 16.0
END DESCRIPTION:
XS GIS Cut Line= 3
      2086525.02     13885975.04      2086475.00     13885875.00
      2086074.95     13885724.98
#Sta/Elev= 30
  4894.3 1197.67  4902.7 1197.11  4953.0 1187.83  4961.4 1184.59  4969.8 1176.83
  4975.4 1173.21  4982.4 1170.94  5008.8 1167.37  5011.3 1166.44  5011.8 1165.94
  5020.6 1166.44  5021.3 1170.41  5027.5 1174.42  5046.2 1176.28  5131.6 1176.02
  5157.2 1177.44  5167.2 1179.46  5186.8 1181.45  5198.4 1183.83  5230.4 1187.92
  5272.3 1197.04  5299.9 1205.70  5326.6 1215.66  5332.8 1218.85  5357.7 1223.90
  5369.3 1228.03  5380.0 1230.68  5388.0 1233.99  5412.0 1239.50  5433.4 1240.90
#Mann=5,-1,0
  4894.3    0.12       0  4982.4    0.07       0  5011.3    0.05       0
  5020.6    0.07       0  5157.2    0.12       0
Bank Sta=5011.3,5020.6
Exp/Cntr=0.3,0.1

Type RM Length L Ch R = 1,6929,432,432,432
BEGIN DESCRIPTION:
GOSS CREEK 15.0
END DESCRIPTION:
XS GIS Cut Line= 3
      2086824.99     13885874.98      2086675.00     13885475.00
      2086724.99     13885275.03
#Sta/Elev= 30
  4576.4 1207.88  4616.4 1198.21  4652.0 1194.69  4683.2 1189.37  4707.2 1187.90
  4732.1 1182.10  4759.9 1179.45  4811.3 1176.21  4832.7 1173.17  4971.5 1171.88
  4982.2 1171.03  5000.9 1165.18  5006.2 1165.18  5008.2 1162.95  5008.3 1162.84
  5008.8 1162.34  5019.5 1162.84  5021.6 1165.49  5026.8 1165.15  5034.5 1167.84
  5044.8 1181.38  5055.1 1186.64  5075.7 1193.54  5109.2 1200.08  5137.6 1211.64
  5150.5 1218.78  5178.8 1227.66  5191.7 1232.80  5207.2 1241.47  5209.7 1241.47
#Mann=5,-1,0
  4576.4    0.12       0  4759.9    0.07       0  5008.2    0.12       0
  5008.3    0.05       0  5019.5    0.12       0
Bank Sta=5008.3,5019.5
Exp/Cntr=0.3,0.1

Type RM Length L Ch R = 1,6497,467,467,467
BEGIN DESCRIPTION:
GOSS CREEK 14.0
END DESCRIPTION:
XS GIS Cut Line= 3
      2086925.00     13885874.99      2087075.00     13885475.00
      2087075.00     13885374.99
#Sta/Elev= 30
  4572.8 1206.54  4575.5 1206.54  4582.6 1203.49  4589.9 1202.50  4604.8 1198.74
  4612.8 1197.77  4618.2 1198.17  4636.9 1195.14  4643.1 1193.10  4690.3 1187.17
  4711.6 1182.76  4743.7 1178.51  4773.9 1176.12  4779.2 1175.63  4814.0 1172.11
  4904.8 1172.08  4967.9 1170.50  4978.6 1169.32  4984.9 1166.54  4990.2 1166.25
  4993.5 1164.66  4997.3 1162.82  5004.4 1162.64  5004.9 1162.14  5015.6 1162.64
  5020.0 1163.90  5030.0 1176.98  5040.0 1186.24  5096.5 1195.27  5100.0 1195.47
#Mann=8,-1,0
  4572.8    0.12       0  4589.9    0.07       0  4773.9   0.035       0
  4779.2    0.07       0  4993.5    0.12       0  5004.4    0.05       0
  5015.6    0.12       0  5096.5    0.07       0
Bank Sta=5004.4,5015.6
Exp/Cntr=0.3,0.1

Type RM Length L Ch R = 1,6030,455,455,455
BEGIN DESCRIPTION:
GOSS CREEK 13.0
END DESCRIPTION:
XS GIS Cut Line= 3
      2087425.00     13885875.01      2087375.00     13885675.00
      2087224.99     13885274.97
#Sta/Elev= 30
  4798.2 1226.73  4821.4 1224.17  4839.4 1214.01  4857.5 1205.75  4898.7 1195.53
  4903.9 1195.70  4928.7 1188.35  4932.2 1187.28  4939.9 1181.54  4945.1 1181.09
  4952.8 1173.34  4963.1 1168.44  4981.2 1161.57  4988.4 1161.00  4988.9 1160.50
  4999.7 1161.00  5001.8 1162.59  5007.0 1162.59  5014.2 1168.56  5068.4 1169.57
  5140.3 1167.42  5165.5 1167.05  5185.0 1168.96  5196.6 1168.73  5215.3 1173.80
  5245.6 1177.86  5275.8 1180.28  5306.1 1186.34  5346.1 1189.25  5431.6 1197.61
#Mann=5,-1,0
  4798.2    0.07       0  4928.7    0.12       0  4988.4    0.05       0
  4999.7    0.12       0  5140.3    0.07       0
Bank Sta=4988.4,4999.7
Exp/Cntr=0.3,0.1

Type RM Length L Ch R = 1,5575,468,468,468
BEGIN DESCRIPTION:
GOSS CREEK 12.0
END DESCRIPTION:
XS GIS Cut Line= 3
      2087825.00     13885625.00      2087725.00     13885475.00
      2087374.99     13885074.99
#Sta/Elev= 30
  4819.7 1223.19  4833.2 1221.56  4863.3 1207.73  4891.8 1197.37  4920.4 1191.60
  4927.9 1188.27  4941.4 1173.53  4950.4 1171.68  4956.4 1166.98  4971.4 1159.63
  4971.8 1157.12  4972.3 1156.62  4983.1 1157.12  4986.5 1157.45  4992.5 1164.10
  4997.0 1165.04  5084.9 1163.76  5134.3 1168.01  5198.8 1166.78  5212.6 1167.34
  5232.6 1171.73  5269.1 1179.40  5290.9 1186.61  5361.1 1195.11  5382.9 1194.61
  5403.8 1198.55  5425.2 1200.26  5446.5 1208.07  5475.0 1213.83  5531.5 1219.41
#Mann=4,-1,0
  4819.7    0.12       0  4971.8    0.05       0  4983.1    0.12       0
  5232.6    0.07       0
Bank Sta=4971.8,4983.1
Exp/Cntr=0.3,0.1

Type RM Length L Ch R = 1,5107,471,471,471
BEGIN DESCRIPTION:
GOSS CREEK 11.0
END DESCRIPTION:
XS GIS Cut Line= 3
      2088123.36     13885658.65      2088025.00     13885125.00
      2087571.26     13884571.83
#Sta/Elev= 30
  4461.8 1204.60  4475.5 1203.57  4480.5 1206.34  4533.6 1197.98  4538.6 1199.79
  4559.2 1197.93  4600.7 1195.36  4619.6 1194.50  4702.7 1189.82  4801.1 1179.73
  4892.6 1165.17  4963.8 1161.48  4972.3 1155.62  4972.8 1155.12  4983.6 1155.62
  4984.1 1157.72  5001.9 1163.45  5056.1 1163.37  5204.6 1163.17  5231.9 1166.28
  5238.4 1169.21  5246.3 1179.74  5444.4 1199.75  5466.6 1206.55  5501.8 1211.72
  5530.5 1219.66  5568.3 1222.81  5643.9 1227.63  5686.9 1238.67  5719.9 1242.78
#Mann=9,-1,0
  4461.8    0.07       0  4559.2    0.12       0  4600.7    0.07       0
  4619.6    0.12       0  4972.3    0.05       0  4983.6    0.12       0
  5056.1   0.035       0  5204.6    0.07       0  5568.3    0.12       0
Bank Sta=4972.3,4983.6
Exp/Cntr=0.3,0.1

Type RM Length L Ch R = 1,4636,468,468,468
BEGIN DESCRIPTION:
GOSS CREEK 10.0
END DESCRIPTION:
XS GIS Cut Line= 3
      2088675.01     13885175.01      2088275.00     13884775.00
      2088109.73     13884371.10
#Sta/Elev= 30
  4438.5 1217.59  4517.7 1200.34  4560.5 1195.55  4622.4 1190.93  4664.8 1185.26
  4735.5 1163.02  4777.9 1160.52  4836.6 1161.08  4848.6 1160.99  4876.9 1164.80
  4891.1 1161.75  4906.9 1161.58  4958.4 1160.15  4961.8 1159.72  4970.1 1153.15
  4970.6 1152.65  4981.8 1153.15  5000.7 1159.32  5018.9 1162.37  5033.0 1177.77
  5036.6 1181.63  5048.3 1184.53  5144.3 1194.33  5155.5 1198.12  5187.9 1201.17
  5227.2 1210.76  5256.6 1220.27  5339.4 1227.32  5393.2 1241.85  5440.6 1245.71
#Mann=9,-1,0
  4438.5    0.12       0  4517.7    0.07       0  4560.5    0.12       0
  4836.6   0.035       0  4906.9    0.07       0  4958.4    0.12       0
  4970.1    0.05       0  4981.8    0.12       0  5033.0    0.07       0
Bank Sta=4970.1,4981.8
Exp/Cntr=0.3,0.1

Type RM Length L Ch R = 1,4168,484,484,484
BEGIN DESCRIPTION:
GOSS CREEK 9.0
END DESCRIPTION:
XS GIS Cut Line= 3
      2088866.43     13885117.04      2088675.00     13884575.00
      2088425.42     13884276.69
#Sta/Elev= 30
  4420.3 1202.42  4485.0 1198.03  4621.0 1188.07  4650.1 1187.47  4681.1 1181.54
  4698.2 1177.60  4719.4 1168.21  4737.6 1162.58  4751.2 1160.06  4831.2 1158.57
  4899.7 1161.16  4963.3 1157.91  4985.0 1157.44  4992.5 1153.22  4998.4 1153.22
  5003.0 1150.40  5003.5 1149.90  5014.7 1150.40  5016.6 1154.79  5066.1 1167.40
  5086.9 1174.92  5094.7 1179.98  5112.8 1184.11  5165.0 1193.62  5222.2 1199.18
  5250.8 1207.73  5257.4 1208.07  5293.8 1221.22  5349.7 1229.29  5384.1 1241.82
#Mann=8,-1,0
  4420.3    0.12       0  4485.0    0.07       0  4621.0    0.12       0
  4831.2   0.035       0  4963.3    0.12       0  5003.0    0.05       0
  5014.7    0.12       0  5112.8    0.07       0
Bank Sta=5003,5014.7
Exp/Cntr=0.3,0.1

Type RM Length L Ch R = 1,3684,487,487,487
BEGIN DESCRIPTION:
GOSS CREEK 8.0
END DESCRIPTION:
XS GIS Cut Line= 3
      2089074.99     13884825.05      2089125.00     13884475.00
      2088775.01     13884075.01
#Sta/Elev= 30
  4646.4 1182.69  4717.2 1176.93  4767.7 1164.86  4798.0 1161.91  4878.8 1157.11
  4939.7 1157.67  4969.7 1156.67  4973.9 1148.02  4974.4 1147.52  4985.7 1148.02
  5006.4 1155.55  5021.5 1156.54  5120.1 1157.73  5162.8 1159.58  5191.2 1162.92
  5212.6 1170.57  5219.7 1181.28  5226.4 1184.65  5311.8 1197.40  5318.9 1199.98
  5332.7 1200.80  5340.3 1205.08  5346.9 1205.63  5373.0 1215.01  5383.0 1219.72
  5397.2 1222.85  5425.2 1225.44  5453.2 1230.91  5481.7 1241.53  5531.5 1245.80
#Mann=7,-1,0
  4646.4    0.12       0  4939.7   0.035       0  4973.9   0.035       0
  4985.7   0.035       0  5006.4    0.12       0  5021.5   0.035       0
  5373.0    0.07       0
Bank Sta=4973.9,4985.7
Exp/Cntr=0.3,0.1

Type RM Length L Ch R = 1,3197,365,365,365
BEGIN DESCRIPTION:
GOSS CREEK 7.0
END DESCRIPTION:
XS GIS Cut Line= 3
      2089296.96     13885096.18      2089575.00     13884375.00
      2088989.59     13883850.39
#Sta/Elev= 30
  4230.6 1202.69  4407.3 1186.96  4478.4 1168.40  4650.7 1159.71  4864.2 1158.00
  4905.7 1153.50  4963.9 1153.77  4976.2 1146.63  4976.7 1146.13  4988.0 1146.63
  5000.8 1153.80  5006.9 1153.80  5010.6 1148.79  5017.3 1155.75  5024.8 1153.26
  5031.5 1160.05  5039.0 1157.52  5045.8 1163.58  5060.0 1166.80  5081.7 1165.28
  5088.4 1170.25  5124.3 1172.87  5131.0 1180.93  5137.8 1182.34  5379.7 1198.00
  5442.7 1200.60  5521.4 1215.28  5584.0 1223.56  5683.5 1228.39  5789.6 1243.28
#Mann=7,-1,0
  4230.6    0.12       0  4650.7   0.035       0  4905.7    0.12       0
  4976.2    0.05       0  4988.0    0.12       0  5379.7   0.035       0
  5521.4    0.07       0
Bank Sta=4976.2,4988
Exp/Cntr=0.3,0.1

Type RM Length L Ch R = 1,2832,650,650,650
BEGIN DESCRIPTION:
GOSS CREEK 6.0
END DESCRIPTION:
XS GIS Cut Line= 4
      2089486.23     13885115.62      2089851.95     13884601.30
      2089779.17     13884391.10      2089025.04     13883794.87
#Sta/Elev= 30
  4368.9 1220.74  4411.3 1212.18  4426.0 1204.46  4432.2 1205.24  4497.4 1189.62
  4547.8 1171.19  4590.5 1162.10  4711.1 1158.69  4934.1 1156.73  4957.2 1153.64
  4978.2 1149.61  5009.0 1150.45  5021.9 1144.22  5022.4 1143.72  5033.7 1144.22
  5049.0 1146.39  5065.4 1154.49  5071.3 1151.88  5091.3 1158.46  5250.8 1163.16
  5321.0 1164.96  5379.0 1168.15  5443.6 1176.59  5508.1 1185.85  5670.9 1195.88
  5814.2 1204.19  5877.9 1217.78  5920.0 1222.45  6062.7 1228.22  6183.8 1243.84
#Mann=11,-1,0
  4368.9    0.12       0  4711.1   0.035       0  4957.2    0.07       0
  5021.9    0.05       0  5033.7    0.07       0  5065.4   0.035       0
  5250.8    0.07       0  5321.0    0.12       0  5379.0    0.07       0
  5443.6    0.12       0  5670.9    0.07       0
Bank Sta=5021.9,5033.7
Exp/Cntr=0.3,0.1

Type RM Length L Ch R = 1,2182,336,336,336
BEGIN DESCRIPTION:
GOSS CREEK 5.0
END DESCRIPTION:
XS GIS Cut Line= 5
      2090186.68     13885162.59      2090289.88     13884754.81
      2090224.82     13884659.91      2089828.64     13884378.31
      2089082.47     13883745.71
#Sta/Elev= 30
  4464.3 1229.56  4565.0 1204.31  4614.9 1196.56  4825.4 1175.40  4833.2 1174.87
  4839.4 1174.32  4901.5 1170.25  4932.5 1168.87  4944.2 1160.18  4989.3 1143.09
  4994.0 1136.76  4994.5 1136.26  5005.9 1136.76  5017.6 1137.50  5024.3 1146.18
  5048.5 1152.98  5068.1 1157.90  5124.6 1160.03  5519.1 1163.80  5577.3 1164.77
  5649.9 1166.27  5732.1 1171.14  5770.7 1181.95  5775.9 1182.43  6086.4 1202.94
  6153.6 1215.18  6214.3 1222.66  6293.5 1225.26  6303.2 1225.43  6464.3 1239.00
#Mann=19,-1,0
  4464.3    0.12       0  4614.9   0.035       0  4825.4    0.12       0
  4833.2   0.035       0  4839.4    0.12       0  4901.5   0.035       0
  4944.2    0.12       0  4994.0    0.05       0  5005.9    0.12       0
  5048.5   0.035       0  5519.1    0.07       0  5577.3   0.035       0
  5649.9    0.07       0  5770.7    0.12       0  5775.9    0.07       0
  6086.4   0.035       0  6153.6    0.07       0  6293.5   0.035       0
  6303.2    0.07       0
Bank Sta=4994,5005.9
Exp/Cntr=0.3,0.1

Type RM Length L Ch R = 1,1846,429,429,429
BEGIN DESCRIPTION:
GOSS CREEK 4.0
END DESCRIPTION:
XS GIS Cut Line= 6
      2090344.84     13885267.34      2090387.20     13884502.99
      2090320.07     13884393.47      2090075.00     13884375.00
      2089916.92     13884352.99      2089169.71     13883760.27
#Sta/Elev= 30
  3865.5 1211.56  3978.0 1191.71  4190.7 1174.53  4256.3 1170.53  4438.7 1166.20
  4598.1 1169.91  4632.5 1170.23  4824.7 1174.03  4864.8 1169.73  4887.0 1163.93
  4922.4 1156.17  4955.1 1147.59  4979.2 1134.37  4979.7 1133.87  4991.1 1134.37
  5007.8 1138.90  5041.0 1157.36  5106.2 1163.99  5414.9 1166.90  5433.7 1168.25
  5477.7 1169.57  5521.0 1182.15  5556.5 1185.52  5744.2 1199.47  5847.8 1204.02
  5891.1 1216.55  5915.4 1220.03  5929.1 1220.69  6027.9 1225.41  6118.6 1228.81
#Mann=16,-1,0
  3865.5    0.12       0  4190.7   0.035       0  4256.3    0.12       0
  4598.1    0.07       0  4632.5    0.12       0  4887.0    0.07       0
  4922.4   0.035       0  4979.2   0.035       0  4991.1   0.035       0
  5414.9    0.07       0  5433.7    0.12       0  5556.5    0.07       0
  5744.2   0.035       0  5915.4    0.07       0  5929.1   0.035       0
  6027.9    0.07       0
Bank Sta=4979.2,4991.1
Exp/Cntr=0.3,0.1

Type RM Length L Ch R = 1,1417,453,453,453
BEGIN DESCRIPTION:
GOSS CREEK 3.0
END DESCRIPTION:
XS GIS Cut Line= 3
      2090178.96     13884026.72      2089925.00     13884025.00
      2089776.14     13884075.33
#Sta/Elev= 30
  4746.0 1174.20  4800.0 1174.01  4819.5 1174.79  4840.0 1173.75  4850.0 1172.04
  4880.0 1168.62  4910.0 1163.61  4940.0 1157.36  4950.0 1154.63  4960.0 1148.76
  4970.0 1139.86  4980.0 1134.95  4990.0 1131.52  4997.5 1128.20  5004.5 1128.05
  5005.0 1127.55  5015.9 1127.55  5016.4 1128.05  5021.1 1132.09  5047.1 1136.19
  5052.7 1139.45  5063.3 1143.42  5073.3 1148.57  5078.6 1150.53  5084.4 1154.15
  5104.7 1159.42  5116.1 1164.06  5126.6 1165.24  5130.4 1165.33  5157.1 1166.69
#Mann=5,-1,0
  4746.0   0.035       0  4819.5    0.07       0  5004.5    0.05       0
  5016.4    0.07       0  5130.4   0.035       0
Bank Sta=5004.5,5016.4
Exp/Cntr=0.3,0.1

Type RM Length L Ch R = 1,964,440,440,440
BEGIN DESCRIPTION:
GOSS CREEK 2.0
END DESCRIPTION:
XS GIS Cut Line= 3
      2090192.80     13883932.93      2090175.00     13883725.00
      2090071.34     13883519.90
#Sta/Elev= 30
  4795.7 1172.35  4813.7 1170.97  4833.8 1171.01  4843.8 1169.13  4873.9 1161.17
  4894.0 1152.52  4904.0 1149.41  4926.0 1145.26  4947.5 1141.78  4954.2 1138.93
  4964.2 1134.24  4974.3 1126.93  4978.3 1122.06  4978.8 1121.56  4990.3 1122.06
  4994.4 1122.89  5001.9 1128.41  5007.2 1128.41  5012.7 1135.81  5018.3 1138.33
  5035.0 1150.08  5040.6 1150.71  5057.3 1159.32  5062.9 1160.43  5079.6 1168.40
  5101.9 1173.68  5124.2 1176.74  5152.1 1178.15  5168.8 1177.29  5234.2 1178.47
#Mann=4,-1,0
  4795.7   0.035       0  4926.0    0.12       0  4978.3    0.05       0
  4990.3    0.12       0
Bank Sta=4978.3,4990.3
Exp/Cntr=0.3,0.1

Type RM Length L Ch R = 1,524,328,328,328
BEGIN DESCRIPTION:
GOSS CREEK 1.0
END DESCRIPTION:
XS GIS Cut Line= 3
      2090609.47     13883853.08      2090575.00     13883625.00
      2090272.65     13883495.46
#Sta/Elev= 30
  4769.1 1160.47  4797.5 1159.82  4827.6 1161.82  4838.0 1160.03  4878.4 1159.46
  4891.0 1156.97  4901.5 1153.21  4929.0 1150.05  4949.2 1143.67  4959.3 1138.27
  4965.3 1132.17  4970.4 1130.06  4979.5 1121.44  4983.7 1115.52  4984.2 1115.02
  4995.7 1115.52  5014.3 1116.92  5021.5 1127.75  5032.4 1132.54  5043.3 1142.61
  5054.2 1146.30  5066.9 1153.32  5085.0 1155.69  5090.4 1157.80  5108.6 1160.71
  5143.0 1161.50  5166.6 1160.67  5213.8 1163.81  5271.8 1163.88  5328.7 1166.95
#Mann=4,-1,0
  4769.1   0.035       0  4891.0    0.12       0  4983.7    0.05       0
  4995.7    0.12       0
Bank Sta=4983.7,4995.7
Exp/Cntr=0.3,0.1

Type RM Length L Ch R = 1,196,0,0,0
BEGIN DESCRIPTION:
GOSS CREEK 0.0
END DESCRIPTION:
XS GIS Cut Line= 3
      2090762.96     13883862.32      2090847.88     13883474.71
      2090354.97     13883199.99
#Sta/Elev= 30
  4603.2 1156.48  4685.1 1155.38  4713.1 1156.83  4778.9 1150.25  4801.5 1148.73
  4815.4 1148.03  4870.7 1136.74  4929.9 1132.41  4948.5 1129.28  4958.4 1124.65
  4963.5 1126.00  4979.2 1115.38  4983.5 1114.89  4984.0 1114.39  4995.5 1114.89
  5009.3 1116.85  5015.1 1123.78  5025.3 1124.01  5031.1 1128.64  5047.1 1130.04
  5052.8 1134.59  5090.5 1141.10  5155.7 1144.32  5177.4 1146.95  5193.4 1151.75
  5215.1 1152.72  5231.1 1155.99  5261.8 1155.93  5268.6 1156.29  5564.3 1154.69
#Mann=8,-1,0
  4603.2   0.035       0  4778.9    0.07       0  4801.5   0.035       0
  4929.9    0.12       0  4983.5    0.05       0  4995.5    0.12       0
  5261.8   0.035       0  5268.6    0.12       0
Bank Sta=4983.5,4995.5
Exp/Cntr=0.3,0.1

Chan Stop Cuts=-1
