--- LITTLE JOSHUA CREEK.prj (project) ---

Proj Title=LITTLE JOSHUA CREEK Base Level Engineering
Current Plan=p01
Default Exp/Contr=0.3,0.1
English Units
Geom File=g01
Flow File=f01
Plan File=p01
Y Axis Title=Elevation
X Axis Title(PF)=Main Channel Distance
X Axis Title(XS)=Station
BEGIN DESCRIPTION:
LITTLE JOSHUA CREEK
END DESCRIPTION:
DSS File=dss
DSS Export Rating Curves= 0
DSS Export Rating Curve Sorted= 0
DSS Export Volume Flow Curves= 0
DXF OffsetX= 0
DXF OffsetY= 0
DXF ScaleX= 1
DXF ScaleY= 10

--- LITTLE JOSHUA CREEK.p01 (plan) ---

Plan Title=Multiple Run
Program Version=4.10
Short Identifier=Multiple Run
Geom File=g01
Flow File=f01
Subcritical Flow
K Sum by GR= 0
Std Step Tol= 0.01
Critical Tol= 0.01
Num of Std Step Trials= 20
Max Error Tol= 0.3
Flow Tol Ratio= 0.001
Split Flow NTrial= 30
Split Flow Tol= 0.02
Split Flow Ratio= 0.02
Log Output Level= 0
Friction Slope Method= 1
Unsteady Friction Slope Method= 2
Unsteady Bridges Friction Slope Method= 1
Parabolic Critical Depth
Global Vel Dist= 1 , 1 , 1
Global Log Level= 0
CheckData=True
Encroach Param=-1 ,0,0, 0
BEGIN DESCRIPTION:
Multiple Run
END DESCRIPTION:
Computation Interval=1HOUR
Output Interval=1HOUR
Run HTab= 0
Run UNet= 0
Run PostProcess= 0
Run WQNet= 0
UNET Theta= 1
UNET Theta Warmup= 1
UNET ZTol= 0.02
UNET ZSATol= 0.05
UNET MxIter= 20
UNET MaxInSteps= 0
UNET DtIC= 0
UNET DtMin= 0
UNET MaxCRTS= 20
UNET WFStab= 2
UNET SFStab= 1
UNET WFX= 1
UNET SFX= 1
UNET DSS MLevel= 4
UNET DZMax Abort= 100
UNET Convert EG Bridges= 0
UNET Use Existing IB Tables=-1
UNET Froude Reduction=False
UNET Froude Limit= 1
UNET Froude Power= 10
UNET Time Slicing=0,0, 5
UNET Junction Losses=0
Instantaneous Interval=1HOUR
DSS File=dss
Write IC File= 0
Write IC File at Sim End=0
Echo Input=False
Echo Parameters=False
Echo Output=False
Write Detailed= 0
WQ AD Non Conservative
WQ ULTIMATE=-1
WQ Max Comp Step=1HOUR
WQ Output Interval=15MIN
WQ Output Selected Increments= 0
WQ Output face flow=0
WQ Output face velocity=0
WQ Output face area=0
WQ Output face dispersion=0
WQ Output cell volume=0
WQ Output cell surface area=0
WQ Output cell continuity=0
WQ Output cumulative cell continuity=0
WQ Output face conc=0
WQ Output face dconc_dx=0
WQ Output face courant=0
WQ Output face peclet=0
WQ Output face adv mass=0
WQ Output face disp mass=0
WQ Output cell mass=0
WQ Output cell source sink temp=0
WQ Output cell source sink nsm=0
WQ Output MaxMinRange=-1
WQ Daily Max Min Mean=-1
WQ Daily Range=0
WQ Daily Time=0
WQ Create Restart=0
WQ Fixed Restart=0
WQ System Summary=0
WQ Use Fixed Temperature=0
Sorting and Armoring Iterations= 10
XS Update Threshold= 0.02
Hydraulics Update Threshold= 0.02
Energy Slope Method= 1
Volume Change Method= 0
XS Weighting Method= 0
Number of US Weighted Cross Sections= 1
Number of DS Weighted Cross Sections= 1
Upstream XS Weight=0.25
Main XS Weight=0.5
Downstream XS Weight=0.25
Number of DS XS's Weighted with US Boundary= 1
Upstream Boundary Weight= 1
Weight of XSs Associated with US Boundary= 0
Number of US XS's Weighted with DS Boundary= 1
Downstream Boundary Weight= 0.5
Weight of XSs Associated with DS Boundary= 0.5
Sediment Output Level= 4
Mass or Volume Output= 0
Output Increment Type= 1
Profile and TS Output Increment= 10
XS Output Flag= 0
XS Output Increment= 10
Disregard all LS=0
Disregard all Conn=0
Disregard all Breaches=0
Disregard all Pumps=0

--- LITTLE JOSHUA CREEK.f01 (steady flow) ---

Flow Title=Multiple
Program Version=4.10
Number of Profiles= 7
Profile Names=10-year,25-year,50-year,1pct_min,100-year,1pct_plu,500-year
River Rch & RM=LITTLE JOSHUA CR,Reach-1         ,44391
     589     965    1312     868    1732    3456    2977
River Rch & RM=LITTLE JOSHUA CR,Reach-1         ,44238
    1289    2226    3134    2139    4269    8517    7834
River Rch & RM=LITTLE JOSHUA CR,Reach-1         ,41139
    2180    3871    5552    3854    7690   15343   14603
River Rch & RM=LITTLE JOSHUA CR,Reach-1         ,37887
    3303    5939    8588    5996   11964   23872   23006
River Rch & RM=LITTLE JOSHUA CR,Reach-1         ,29008
    3717    6703    9711    6790   13548   27031   26121
River Rch & RM=LITTLE JOSHUA CR,Reach-1         ,24739
    3915    7071   10255    7176   14318   28568   27652
River Rch & RM=LITTLE JOSHUA CR,Reach-1         ,22313
    5575   10167   14843   10445   20841   41584   40693
River Rch & RM=LITTLE JOSHUA CR,Reach-1         ,16220
    5715   10414   15196   10686   21320   42540   41567
River Rch & RM=LITTLE JOSHUA CR,Reach-1         ,12005
    5872   10705   15624   10989   21925   43747   42760
River Rch & RM=LITTLE JOSHUA CR,Reach-1         ,10933
    8154   15047   22147   15695   31317   62485   62005
River Rch & RM=LITTLE JOSHUA CR,Reach-1         ,9270
    8195   15087   22170   15683   31293   62437   61734
River Rch & RM=LITTLE JOSHUA CR,Reach-1         ,4400
    8501   15646   22986   16253   32430   64706   63921
Boundary for River Rch & Prof#=LITTLE JOSHUA CR,Reach-1         , 1
Up Type= 0
Dn Type= 1
Dn Known WS=1333.57
Boundary for River Rch & Prof#=LITTLE JOSHUA CR,Reach-1         , 2
Up Type= 0
Dn Type= 1
Dn Known WS=1337.31
Boundary for River Rch & Prof#=LITTLE JOSHUA CR,Reach-1         , 3
Up Type= 0
Dn Type= 1
Dn Known WS=1340.46
Boundary for River Rch & Prof#=LITTLE JOSHUA CR,Reach-1         , 4
Up Type= 0
Dn Type= 1
Dn Known WS=1337.64
Boundary for River Rch & Prof#=LITTLE JOSHUA CR,Reach-1         , 5
Up Type= 0
Dn Type= 1
Dn Known WS=1343.85
Boundary for River Rch & Prof#=LITTLE JOSHUA CR,Reach-1         , 6
Up Type= 0
Dn Type= 1
Dn Known WS=1348.2
Boundary for River Rch & Prof#=LITTLE JOSHUA CR,Reach-1         , 7
Up Type= 0
Dn Type= 1
Dn Known WS=1348.17
DSS Import GetInterval= 0
DSS Import GetPeak= 0
DSS Import FillOption= 0

--- LITTLE JOSHUA CREEK.g01 (geometry) ---

Geom Title=Existing Conditions
Program Version=4.10

River Reach=LITTLE JOSHUA CR,Reach-1
Reach XY= 30
        2020075.       13860125.       2018982.2      13862675.3
       2019673.8      13863685.5        2019375.       13864775.
      2020222.95     13865180.84      2020101.14     13866401.94
      2020919.74     13866580.47      2021271.86      13867467.5
      2021554.86     13866774.59      2021872.71     13867619.88
      2022981.19     13867532.82      2025052.01     13868951.48
      2025071.38     13869667.51      2025926.68     13869028.08
      2026164.29      13869324.3      2027240.16     13868825.39
      2027976.56     13869521.26      2028681.15     13869331.94
      2029518.84     13870817.22      2031658.59      13871258.2
      2031918.81     13872917.19      2032969.82     13872380.41
      2034532.86     13875081.19      2035617.14     13876018.83
      2035566.76     13877228.23      2034624.61       13879050.
      2035474.48     13881840.22      2035458.57     13882391.77
      2034575.38     13882840.16        2035175.       13884075.

Type RM Length L Ch R = 1 ,44391   ,154,154,154
BEGIN DESCRIPTION:
LITTLE JOSHUA CREEK 90.0
END DESCRIPTION:
XS GIS Cut Line= 3
      2019829.66     13859947.81      2020074.62     13860137.96
      2020510.07     13859942.26
#Sta/Elev= 30
  4689.9 1779.75  4691.9 1777.59  4727.2 1772.13  4770.7 1757.59  4791.5 1754.92
  4812.3  1742.7  4841.2 1741.43  4862.1 1735.83  4884.7 1725.97  4905.5 1722.79
    4920 1712.72  4940.8 1709.02    4949 1702.97  4955.3 1703.08  4969.8 1689.83
  4976.1 1689.11  4984.3 1683.49  5009.4 1680.61  5009.6 1680.11  5013.4 1680.61
  5099.1 1691.95  5162.6 1694.64  5252.6 1702.48  5283.9 1709.69  5312.5 1713.07
  5335.7    1721  5387.5 1730.19  5433.8 1744.17  5462.4 1748.97  5477.4 1755.57
#Mann= 3 ,-1 , 0
  4689.9     .12       0  5009.4     .05       0  5013.4     .12       0
Bank Sta=5009.4,5013.4
XS Rating Curve= 0 ,0
Exp/Cntr=0.3,0.1

Type RM Length L Ch R = 1 ,44238   ,447,447,447
BEGIN DESCRIPTION:
LITTLE JOSHUA CREEK 89.0
END DESCRIPTION:
XS GIS Cut Line= 3
      2019674.76     13860157.65        2020125.       13860275.
       2020630.4     13860363.08
#Sta/Elev= 30
  4534.3 1757.22  4541.7 1757.11  4546.8 1752.79  4575.9 1753.39  4582.2 1752.64
  4587.3 1748.94  4720.6 1736.69  4744.1 1727.51  4860.4 1702.03  4968.6 1687.47
  4976.7 1684.42  4989.2 1685.48  5017.9 1680.35  5018.1 1679.85  5021.9 1680.35
  5060.7 1680.94  5121.4 1682.29  5140.9  1695.1  5172.1 1701.38    5233 1710.84
  5253.3 1711.66  5283.8 1719.26  5319.6 1722.99  5344.7 1728.35  5367.4 1728.46
  5425.9 1732.08  5433.7 1733.53  5438.8  1737.9  5476.7 1737.56  5512.6 1747.07
#Mann= 5 ,-1 , 0
  4534.3     .12       0  5017.9     .05       0  5021.9     .12       0
  5060.7     .07       0  5367.4     .12       0
Bank Sta=5017.9,5021.9
XS Rating Curve= 0 ,0
Exp/Cntr=0.3,0.1

Type RM Length L Ch R = 1 ,43791   ,423,423,423
BEGIN DESCRIPTION:
LITTLE JOSHUA CREEK 88.0
END DESCRIPTION:
XS GIS Cut Line= 3
      2019825.02     13860425.03        2019925.       13860625.
        2020225.       13860725.
#Sta/Elev= 30
  4776.4 1706.39  4790.3 1704.83  4807.1 1700.61  4812.7 1700.51  4829.5 1694.61
  4835.1 1694.03  4851.8 1684.39  4874.2 1677.16  4896.6 1673.33  4941.3 1671.13
  4946.9  1671.6  4991.6 1668.57  4997.2 1666.33  5002.6 1666.33  5010.5 1664.26
  5019.1 1664.15  5019.3 1663.65  5023.1 1664.15  5042.1 1665.36  5052.7 1675.49
  5063.2 1678.51  5084.3 1681.89  5115.9 1684.53    5137 1685.15  5200.2 1693.88
  5221.3 1698.79  5242.4 1705.13  5284.6 1713.72  5313.6 1723.59  5316.2 1723.59
#Mann= 3 ,-1 , 0
  4776.4     .12       0  5019.1     .05       0  5023.1     .12       0
Bank Sta=5019.1,5023.1
XS Rating Curve= 0 ,0
Exp/Cntr=0.3,0.1

Type RM Length L Ch R = 1 ,43368   ,446,446,446
BEGIN DESCRIPTION:
LITTLE JOSHUA CREEK 87.0
END DESCRIPTION:
XS GIS Cut Line= 3
      2019374.98       13860875.        2019675.       13860925.
        2019975.       13860975.
#Sta/Elev= 30
  4691.2 1728.82  4693.8 1728.82  4701.4 1724.76  4711.5 1723.21  4724.2 1719.74
  4741.9 1710.64  4802.7 1697.81    4823 1691.61  4833.2 1690.16  4840.8 1686.42
  4863.6 1683.58  4901.6 1674.99  4906.7  1675.5  4924.4 1670.43  4934.5 1664.91
  4944.7 1662.89  4960.4 1658.23  4960.7 1657.73  4964.4 1658.23  4967.5 1659.31
  4997.9 1658.44  5015.6 1661.59  5023.2 1662.29  5028.3 1661.54  5056.2 1663.85
  5084.1 1664.41  5106.9 1663.97    5150 1668.03  5218.4 1676.23  5299.5 1682.57
#Mann= 3 ,-1 , 0
  4691.2     .12       0  4960.4     .05       0  4964.4     .12       0
Bank Sta=4960.4,4964.4
XS Rating Curve= 0 ,0
Exp/Cntr=0.3,0.1

Type RM Length L Ch R = 1 ,42922   ,442,442,442
BEGIN DESCRIPTION:
LITTLE JOSHUA CREEK 86.0
END DESCRIPTION:
XS GIS Cut Line= 3
      2019674.98     13861224.98        2019725.       13861275.
      2019874.99     13861374.99
#Sta/Elev= 30
  4924.8 1668.34  4953.1 1666.73  4967.2 1665.16  4981.4  1661.2    4992 1650.87
  4998.5 1650.87    5003  1648.4  5007.1 1647.77  5007.3 1647.27  5010.8 1647.27
  5011.1 1647.77  5024.1 1648.35  5031.6 1651.72  5039.1 1653.78  5045.1 1652.14
  5054.1 1657.19  5060.1 1655.88  5067.6  1659.3  5075.2 1659.58  5090.2 1662.13
  5103.7 1663.04  5111.2 1664.65  5117.2 1667.51  5126.2 1669.72  5132.2 1672.76
  5139.8 1674.29  5162.3 1675.97  5168.3 1675.92  5172.8 1676.99  5175.8 1676.99
#Mann= 3 ,-1 , 0
  4924.8     .12       0  5007.1     .05       0  5011.1     .12       0
Bank Sta=5007.1,5011.1
XS Rating Curve= 0 ,0
Exp/Cntr=0.3,0.1

Type RM Length L Ch R = 1 ,42480   ,484,484,484
BEGIN DESCRIPTION:
LITTLE JOSHUA CREEK 85.0
END DESCRIPTION:
XS GIS Cut Line= 3
      2019201.87     13861462.38        2019475.       13861625.
      2019990.93     13861757.31
#Sta/Elev= 30
  4677.9 1703.35  4704.8  1700.9  4711.5 1698.98  4717.3 1695.48  4797.9 1679.96
  4806.9 1680.29  4849.7 1674.93  4865.3 1670.84  4886.7 1670.78  4892.6 1669.26
  4908.2 1668.44  4937.6 1664.41    4988  1653.2  4992.9 1648.83  4998.4 1648.83
  5006.1 1643.71  5011.6 1641.55  5011.8 1641.05  5015.6 1641.55  5018.7 1641.63
  5054.4 1652.09  5078.4 1655.43  5176.7 1662.36  5367.4 1673.08  5398.4 1676.19
  5439.7 1683.25  5462.1 1685.88  5502.9 1696.65  5522.3    1703  5528.4 1706.08
#Mann= 3 ,-1 , 0
  4677.9     .12       0  5011.6     .05       0  5015.6     .12       0
Bank Sta=5011.6,5015.6
XS Rating Curve= 0 ,0
Exp/Cntr=0.3,0.1

Type RM Length L Ch R = 1 ,41996   ,415,415,415
BEGIN DESCRIPTION:
LITTLE JOSHUA CREEK 84.0
END DESCRIPTION:
XS GIS Cut Line= 3
      2019225.02     13861775.02      2019488.34     13862048.33
      2019844.23     13862143.81
#Sta/Elev= 30
  4608.4 1681.22  4643.1 1677.85  4664.8 1672.07  4686.2 1668.86  4735.6 1663.47
  4905.4 1649.39  4926.7 1646.33  4947.8 1645.88  4976.1 1638.75  4987.9  1637.9
    4990 1635.52  4990.3 1635.02    4994 1635.52  5005.2 1636.72  5015.5 1641.47
  5025.2 1649.85    5032 1653.82  5037.2 1653.42  5045.9 1656.99  5129.4 1667.75
  5170.8 1676.24  5201.9  1680.3  5221.7 1685.93  5226.8 1685.38    5233 1688.24
  5242.1  1689.5  5274.4 1691.81  5295.1 1695.36  5326.1 1703.44  5356.4 1707.81
#Mann= 6 ,-1 , 0
  4608.4     .12       0    4990     .05       0    4994     .12       0
  5025.2    .035       0  5045.9     .07       0  5242.1     .12       0
Bank Sta=4990,4994
XS Rating Curve= 0 ,0
Exp/Cntr=0.3,0.1

Type RM Length L Ch R = 1 ,41581   ,442,442,442
BEGIN DESCRIPTION:
LITTLE JOSHUA CREEK 83.0
END DESCRIPTION:
XS GIS Cut Line= 3
      2019019.59      13861926.8        2019125.       13862175.
      2020136.39     13862230.95
#Sta/Elev= 30
  4734.9 1687.95  4784.5 1679.62  4813.6 1677.73  4837.2 1669.25    4890 1664.28
  4937.3 1650.52    4972 1637.32  5001.8 1631.16  5012.6 1630.45  5012.8 1629.95
  5016.6 1630.45  5074.7 1641.79  5160.8 1648.88  5247.7 1653.44  5458.7  1664.7
  5516.5 1671.02  5611.4 1686.37  5634.4 1690.52  5639.4 1689.46  5675.6 1694.66
  5715.6 1701.72  5735.7 1706.27  5775.7 1719.39  5845.8 1725.39  5875.9 1731.99
    5916    1737    5946 1742.76  5995.7 1747.64  6000.7 1744.09  6017.5 1745.34
#Mann= 7 ,-1 , 0
  4734.9     .12       0  5012.6     .05       0  5016.6     .12       0
  5160.8     .07       0  5247.7    .035       0  5516.5     .07       0
  5611.4     .12       0
Bank Sta=5012.6,5016.6
XS Rating Curve= 0 ,0
Exp/Cntr=0.3,0.1

Type RM Length L Ch R = 1 ,41139   ,460,460,460
BEGIN DESCRIPTION:
LITTLE JOSHUA CREEK 82.0
END DESCRIPTION:
XS GIS Cut Line= 3
      2018672.33     13862534.45        2019075.       13862475.
      2020108.98     13862621.24
#Sta/Elev= 30
  4588.2 1665.35  4793.1 1649.82  4821.2 1641.44  4873.9 1635.92  4924.5 1636.45
  4944.7 1635.96  4960.4 1633.23  4965.5 1634.32  4992.7 1626.57  5002.7 1625.64
  5003.1 1625.14    5008 1625.64  5045.7 1627.03  5055.8 1638.07  5065.9 1644.44
  5171.5  1650.4  5298.2 1651.46  5328.5 1647.83    5386 1651.88  5448.2 1651.66
  5462.1 1654.66  5525.5 1657.83  5540.6 1662.39  5604.2 1668.54  5712.3  1675.7
  5843.6 1687.91  5945.8 1701.28  5959.5 1704.79  6015.3 1709.69  6039.5 1716.09
#Mann= 6 ,-1 , 0
  4588.2     .12       0  5002.7     .05       0    5008     .12       0
  5171.5     .07       0  5448.2     .12       0  5945.8     .07       0
Bank Sta=5002.7,5008
XS Rating Curve= 0 ,0
Exp/Cntr=0.3,0.1

Type RM Length L Ch R = 1 ,40679   ,484,484,484
BEGIN DESCRIPTION:
LITTLE JOSHUA CREEK 81.0
END DESCRIPTION:
XS GIS Cut Line= 3
      2018711.44     13862877.32        2019125.       13862825.
      2019691.12     13862647.67
#Sta/Elev= 30
  4582.7 1674.75  4626.6 1668.13  4838.3    1648  4858.4 1645.12  4868.5 1642.51
  4876.8 1637.25  4881.8 1632.35  4888.7 1628.54    4957 1627.75  4994.3 1625.65
  4994.7 1625.15  4999.8 1625.65  5015.8 1627.75    5021 1626.65  5048.2 1633.03
  5053.5 1630.82  5080.7 1633.87  5085.9 1630.47  5113.1 1635.88  5118.4 1633.66
  5125.3 1636.01  5145.6 1637.84  5150.8 1636.75  5187.5 1642.43  5230.1  1647.6
  5303.4 1651.65  5411.7 1661.06  5502.5 1668.45  5550.6 1673.72  5592.8 1675.87
#Mann= 5 ,-1 , 0
  4582.7     .12       0  4994.3     .05       0  4999.8     .12       0
  5187.5     .07       0  5411.7     .12       0
Bank Sta=4994.3,4999.8
XS Rating Curve= 0 ,0
Exp/Cntr=0.3,0.1

Type RM Length L Ch R = 1 ,40195   ,439,439,439
BEGIN DESCRIPTION:
LITTLE JOSHUA CREEK 80.0
END DESCRIPTION:
XS GIS Cut Line= 3
      2018925.02       13863225.        2019325.       13863225.
      2019675.01     13862824.99
#Sta/Elev= 30
  4584.6 1654.32  4614.6 1651.29  4668.8 1647.63  4767.4 1641.13  4874.6 1633.91
  4904.6 1629.04  4934.6 1628.17  4944.6 1627.53  4954.6  1625.7  4964.5 1625.38
  4973.9 1625.36  4988.9 1625.36  4989.4 1624.86  4994.4 1625.36  5083.8 1625.64
    5098 1628.54  5118.9 1630.91  5183.4 1640.14  5210.9 1645.04  5218.5 1645.19
  5253.7 1650.35  5280.5 1653.43  5303.5 1656.03  5402.2  1664.2  5437.8 1668.24
  5466.3 1670.27  5488.1    1673  5494.7 1675.21    5509 1676.99  5516.1 1676.96
#Mann= 8 ,-1 , 0
  4584.6    .035       0  4668.8     .07       0  4767.4     .12       0
  4964.5     .07       0  4973.9     .12       0  4988.9     .05       0
  4994.4     .12       0  5280.5     .07       0
Bank Sta=4988.9,4994.4
XS Rating Curve= 0 ,0
Exp/Cntr=0.3,0.1

Type RM Length L Ch R = 1 ,39931   ,175,175,175
BEGIN DESCRIPTION:
LITTLE JOSHUA CREEK 79.5
END DESCRIPTION:
XS GIS Cut Line= 4
       2018791.6     13863453.93      2019433.76     13863290.03
      2019558.99     13863258.04      2019956.83     13863108.25
#Sta/Elev= 30
    4208 1664.45  4411.4 1648.99  4424.6 1647.23  4493.9 1644.23  4628.9 1637.76
  4705.4 1628.45  4710.6 1630.21  4737.1 1631.91  4787.2 1633.41  4799.8 1631.86
  4837.1 1632.06  4909.7 1630.92  4982.8 1625.91  4983.2 1625.41  4988.3 1625.91
  5017.1 1627.92    5028 1631.17  5043.8 1632.57  5052.9 1634.34  5077.7 1643.21
  5102.6 1644.83  5150.3  1654.8  5198.8 1661.14  5241.5 1664.01  5324.4 1672.68
  5366.5 1678.86  5394.1 1682.25  5412.5 1685.76    5419 1688.36  5425.1 1688.23
#Mann= 11 ,-1 , 0
    4208     .12       0  4411.4    .035       0  4493.9     .12       0
  4737.1     .07       0  4837.1     .12       0  4982.8     .05       0
  4988.3     .12       0  5043.8     .07       0  5150.3     .12       0
  5324.4     .07       0  5366.5     .12       0
Bank Sta=4982.8,4988.3
XS Rating Curve= 0 ,0
Exp/Cntr=0.3,0.1

Type RM Length L Ch R = 1 ,39756   ,470,470,470
BEGIN DESCRIPTION:
LITTLE JOSHUA CREEK 79.0
END DESCRIPTION:
XS GIS Cut Line= 3
      2018993.52     13863662.93        2019475.       13863375.
       2019949.6     13863229.85
#Sta/Elev= 30
  4435.4 1661.84  4469.6 1659.81  4548.9 1653.91  4659.9 1641.12  4727.3 1635.63
  4829.1 1630.39  4844.7 1628.74  4850.5 1624.55  4871.9 1623.13  4924.4  1624.6
  4930.3 1623.61  4938.1 1618.86  4945.8 1610.37  4961.4 1603.27  4982.8  1604.5
    5004  1602.6  5004.5  1602.1  5009.7  1602.6    5018 1603.65  5029.4 1612.83
  5050.8 1630.86  5059.1  1632.1  5078.4 1626.06    5101 1625.77  5132.3 1627.62
    5141 1630.17  5174.2 1640.07    5228 1645.05  5446.2 1668.34  5492.7 1675.64
#Mann= 10 ,-1 , 0
  4435.4     .12       0  4469.6     .07       0  4548.9     .12       0
  4727.3     .07       0    5004     .05       0  5009.7     .07       0
  5029.4     .12       0    5141     .07       0    5228     .12       0
  5446.2     .07       0
Bank Sta=5004,5009.7
XS Rating Curve= 0 ,0
Exp/Cntr=0.3,0.1

Type RM Length L Ch R = 1 ,39286   ,499,499,499
BEGIN DESCRIPTION:
LITTLE JOSHUA CREEK 78.0
END DESCRIPTION:
XS GIS Cut Line= 3
      2019371.13      13863780.1        2019675.       13863775.
      2020111.68     13863775.76
#Sta/Elev= 30
    4696 1634.06  4703.5  1634.2  4719.9 1632.55  4759.9 1626.87  4829.9 1621.42
  4849.9 1620.64  4879.9 1614.94  4902.3 1612.38  4919.9 1609.99  4939.9 1602.01
  4959.9 1599.74  4969.9 1600.12  4979.9 1599.53  4997.4  1595.5    5007  1595.3
  5007.5  1594.8  5012.9  1595.3  5019.9 1597.82  5029.9 1610.58  5039.9 1622.18
  5059.9 1622.06  5109.9 1623.44  5149.9 1625.93  5219.9  1633.1  5239.9 1634.56
  5279.9  1639.9  5329.9 1650.38  5389.9 1658.19  5413.9 1660.34  5436.6 1662.05
#Mann= 5 ,-1 , 0
    4696     .07       0  4902.3     .12       0    5007     .05       0
  5012.9     .12       0  5413.9     .07       0
Bank Sta=5007,5012.9
XS Rating Curve= 0 ,0
Exp/Cntr=0.3,0.1

Type RM Length L Ch R = 1 ,38787   ,377,377,377
BEGIN DESCRIPTION:
LITTLE JOSHUA CREEK 77.0
END DESCRIPTION:
XS GIS Cut Line= 3
      2019175.84     13864105.62        2019675.       13864275.
      2020011.77     13864266.26
#Sta/Elev= 30
  4472.5  1627.4  4481.5 1626.94  4486.8 1625.05  4544.3 1620.75  4556.1 1618.37
  4587.8  1615.8  4651.1 1611.29  4693.4  1609.6  4800.8  1609.5  4915.1 1612.82
  4920.4 1612.21  4936.3 1604.48  4946.8 1597.17  4952.5 1595.22  4957.8 1595.77
  4978.5 1588.11  4986.2 1587.76  4986.7 1587.26  4992.1 1587.76    4997 1590.17
  5009.6 1591.82  5029.6 1597.74  5039.6 1604.98  5059.6 1612.33  5179.7 1619.58
  5229.7 1625.21  5239.7 1628.55  5269.7 1645.87  5279.7 1648.24  5336.5 1655.12
#Mann= 3 ,-1 , 0
  4472.5     .12       0  4986.2     .05       0  4992.1     .12       0
Bank Sta=4986.2,4992.1
XS Rating Curve= 0 ,0
Exp/Cntr=0.3,0.1

Type RM Length L Ch R = 1 ,38410   ,523,523,523
BEGIN DESCRIPTION:
LITTLE JOSHUA CREEK 76.0
END DESCRIPTION:
XS GIS Cut Line= 3
      2018989.25      13864457.2      2019536.08     13864609.09
      2019791.06     13864578.84
#Sta/Elev= 30
  4426.3 1651.32  4437.1 1651.59    4453 1649.02  4471.4 1641.81  4476.6 1644.88
  4504.9 1632.25  4510.8 1627.73    4516 1631.02  4545.1 1616.88  4550.2 1618.48
  4567.2 1608.62  4577.6 1606.52  4623.9  1603.7  4681.4 1603.51  4743.6 1608.62
  4816.3 1606.54    4837 1602.41  4857.8 1591.84  4889.6 1589.52  4951.2  1588.8
  4982.3 1585.49  4987.7 1582.39  4988.2 1581.89  4993.6 1582.39  5002.8 1582.47
  5012.9 1586.53    5033 1599.63  5043.1 1604.34  5143.8 1606.65  5250.6 1612.32
#Mann= 3 ,-1 , 0
  4426.3     .12       0  4987.7     .05       0  4993.6     .12       0
Bank Sta=4987.7,4993.6
XS Rating Curve= 0 ,0
Exp/Cntr=0.3,0.1

Type RM Length L Ch R = 1 ,37887   ,465,465,465
BEGIN DESCRIPTION:
LITTLE JOSHUA CREEK 75.0
END DESCRIPTION:
XS GIS Cut Line= 3
      2019214.91     13865364.29        2019625.       13864825.
      2019900.31     13864522.68
#Sta/Elev= 30
  4326.8 1613.78  4361.4 1611.96  4565.7 1605.42  4697.6 1603.26  4803.7 1599.94
  4826.5 1600.18  4868.1 1595.69  4890.9 1590.26  4924.6 1587.73  4954.1 1582.04
  4961.7 1578.29    4978 1576.97  4978.5 1576.47    4987 1576.97    4997 1577.38
  5001.2 1581.58  5007.7 1581.58  5011.4 1583.11  5018.2 1582.92  5025.6 1587.58
  5032.3 1589.07  5039.8 1592.79  5046.5 1592.81    5054  1595.3  5131.7 1598.68
  5237.8 1605.94  5308.7  1612.6  5343.8 1617.72  5372.2    1624  5413.2 1628.27
#Mann= 6 ,-1 , 0
  4326.8     .07       0  4361.4    .035       0  4565.7     .07       0
  4924.6     .12       0    4978     .05       0    4987     .12       0
Bank Sta=4978,4987
XS Rating Curve= 0 ,0
Exp/Cntr=0.3,0.1

Type RM Length L Ch R = 1 ,37422   ,459,459,459
BEGIN DESCRIPTION:
LITTLE JOSHUA CREEK 74.0
END DESCRIPTION:
XS GIS Cut Line= 3
      2019475.36     13865329.56        2020025.       13865025.
      2020225.02     13864874.99
#Sta/Elev= 30
  4377.7 1603.26    4499 1599.17  4623.7 1598.21  4674.5 1599.15  4764.5  1593.5
  4889.3 1592.57    4895 1590.08  4911.1 1589.37  4916.8 1586.32  4940.6 1580.84
  4970.6 1580.86  4992.3 1573.72  4993.6 1572.15  4994.1 1571.65  5002.6 1572.15
  5019.6 1572.63  5034.2 1579.11  5042.5  1580.3  5048.8 1584.25  5092.5 1587.63
  5113.4 1597.86  5134.2 1613.06  5142.5 1615.58  5148.8 1619.87  5169.6 1630.28
  5184.2 1636.37  5213.4 1652.71  5248.8 1658.51    5253 1660.73  5256.1 1660.73
#Mann= 4 ,-1 , 0
  4377.7     .07       0  4940.6     .12       0  4993.6     .05       0
  5002.6     .12       0
Bank Sta=4993.6,5002.6
XS Rating Curve= 0 ,0
Exp/Cntr=0.3,0.1

Type RM Length L Ch R = 1 ,36963   ,465,465,465
BEGIN DESCRIPTION:
LITTLE JOSHUA CREEK 73.0
END DESCRIPTION:
XS GIS Cut Line= 3
      2019501.31     13865420.73        2020225.       13865375.
      2020374.96     13865424.99
#Sta/Elev= 30
  4279.6 1602.52  4393.5 1597.59  4463.7 1596.55  4483.7 1594.26  4513.8 1592.91
  4603.6 1590.74  4768.1 1590.29  4814.4 1589.21  4824.2 1588.03  4844.4  1583.5
  4864.5  1580.9  4944.6  1577.9  4964.6 1573.76  4974.7 1570.19  4990.2  1568.9
  4990.7  1568.4  4999.3  1568.9  5002.2 1573.53  5007.4 1573.53  5015.3  1576.1
  5046.9 1596.48  5057.4 1599.63  5078.5 1608.43  5083.8 1612.44  5089.1 1612.02
  5110.1 1626.39  5120.7 1631.76  5131.2  1638.5  5141.8 1643.19  5162.8 1646.36
#Mann= 4 ,-1 , 0
  4279.6     .07       0  4824.2     .12       0  4990.2     .05       0
  4999.3     .12       0
Bank Sta=4990.2,4999.3
XS Rating Curve= 0 ,0
Exp/Cntr=0.3,0.1

Type RM Length L Ch R = 1 ,36498   ,483,483,483
BEGIN DESCRIPTION:
LITTLE JOSHUA CREEK 72.0
END DESCRIPTION:
XS GIS Cut Line= 3
       2019358.1     13865846.07        2020175.       13865825.
      2020474.98     13865625.01
#Sta/Elev= 30
  4182.8 1607.98  4199.7 1604.29  4239.7 1602.89  4299.7 1594.66  4416.6 1585.58
  4499.8 1582.33  4699.9 1582.95  4839.9 1587.29  4885.5 1586.43  4929.9 1583.73
    4960 1572.88  4992.9 1565.77  4993.4 1565.27  5002.1 1565.77  5043.5 1574.47
  5064.6 1575.63  5144.2 1586.75  5151.7 1589.33  5157.7 1593.97  5172.7 1595.06
  5208.8 1608.76  5223.8 1609.33  5229.8 1612.88  5238.8 1613.76  5280.9 1630.53
  5301.9 1636.05  5310.9 1635.94    5332 1641.04    5338 1644.23  5360.5 1647.94
#Mann= 4 ,-1 , 0
  4182.8     .07       0  4885.5     .12       0  4992.9     .05       0
  5002.1     .12       0
Bank Sta=4992.9,5002.1
XS Rating Curve= 0 ,0
Exp/Cntr=0.3,0.1

Type RM Length L Ch R = 1 ,36015   ,168,168,168
BEGIN DESCRIPTION:
LITTLE JOSHUA CREEK 71.0
END DESCRIPTION:
XS GIS Cut Line= 3
      2019483.97     13866392.95        2020075.       13866275.
      2020475.02     13865874.98
#Sta/Elev= 30
  4397.8 1605.91  4408.4 1605.88  4419.2  1607.5  4429.4 1603.75  4449.8 1598.01
  4470.2  1593.1  4490.6 1589.55  4521.2 1585.01  4572.2 1580.97  4653.8 1577.75
  4896.8 1575.51  4923.9 1575.17  4959.7 1570.14  4969.9 1570.64  4990.3 1566.26
    5004 1565.46    5010 1563.23  5010.5 1562.73  5019.2 1563.23  5028.8 1563.81
  5042.9 1566.53  5057.1 1567.92  5085.3    1574  5113.6 1577.81    5255 1576.06
  5311.6 1576.39    5354 1577.79  5467.2 1583.01  5509.6 1586.62  5566.2 1594.18
#Mann= 4 ,-1 , 0
  4397.8     .07       0  4896.8     .12       0    5010     .05       0
  5019.2     .12       0
Bank Sta=5010,5019.2
XS Rating Curve= 0 ,0
Exp/Cntr=0.3,0.1

Type RM Length L Ch R = 1 ,35847   ,808,808,808
BEGIN DESCRIPTION:
LITTLE JOSHUA CREEK 70.0
END DESCRIPTION:
XS GIS Cut Line= 3
      2019280.83     13867130.86      2020124.65     13866425.35
      2020774.99     13866075.01
#Sta/Elev= 30
  3900.1 1680.33  4013.4 1664.58  4219.1 1642.67  4418.2 1623.79  4564.2 1616.62
    4602    1608  4773.4 1591.25    4802 1591.79  4837.2 1601.24  4886.6 1600.58
  4936.1 1592.69  4958.2 1567.77  4974.4 1559.94  4974.9 1559.44  4983.7 1559.94
  5014.4 1567.04  5058.2 1570.21  5533.5 1574.32  5577.3 1586.54    5583 1592.42
  5599.2 1595.04  5604.9 1603.24  5621.1 1602.98  5626.8 1609.82    5643 1612.14
  5648.7 1619.69  5664.9 1623.53  5670.6 1631.52  5686.8 1640.12  5738.7 1654.04
#Mann= 5 ,-1 , 0
  3900.1     .07       0  4564.2    .035       0    4602     .12       0
  4974.4     .05       0  4983.7     .12       0
Bank Sta=4974.4,4983.7
XS Rating Curve= 0 ,0
Exp/Cntr=0.3,0.1

Type RM Length L Ch R = 1 ,35039   ,473,473,473
BEGIN DESCRIPTION:
LITTLE JOSHUA CREEK 69.0
END DESCRIPTION:
XS GIS Cut Line= 3
      2020087.33     13866909.43        2020875.       13866575.
      2021174.98     13866175.02
#Sta/Elev= 30
  4139.4 1604.37  4256.4 1599.07  4451.9 1586.16    4604 1580.13  4698.6 1572.91
  4712.7 1574.68    4775  1566.8  4962.5 1562.63  4973.4 1561.79  4992.4 1556.13
  5018.5 1553.33    5019 1552.83  5028.1 1553.33  5037.8 1561.79  5045.1 1564.02
  5081.9 1567.33  5152.4 1573.23  5202.4 1581.34    5217 1586.84  5231.6 1594.92
  5237.8 1600.49  5258.7    1610    5267 1611.24  5287.8 1627.35  5295.1 1630.02
  5423.3 1662.24    5467 1678.23  5487.8 1683.06    5492 1687.33  5495.1 1687.33
#Mann= 4 ,-1 , 0
  4139.4    .035       0  5018.5    .035       0  5028.1    .035       0
  5081.9     .12       0
Bank Sta=5018.5,5028.1
XS Rating Curve= 0 ,0
Exp/Cntr=0.3,0.1

Type RM Length L Ch R = 1 ,34566   ,327,327,327
BEGIN DESCRIPTION:
LITTLE JOSHUA CREEK 68.0
END DESCRIPTION:
XS GIS Cut Line= 3
      2020412.81      13867421.6        2021025.       13866975.
      2021425.02     13866574.98
#Sta/Elev= 30
  4246.5 1603.38  4323.5 1599.84  4352.7 1596.24  4453.1  1588.1  4538.9 1583.43
  4553.6 1581.57  4674.8 1575.88  4710.4  1575.1  4718.9 1576.19    4725 1575.75
  4740.8 1571.36  4799.9 1563.69  4925.9 1557.95  4954.8 1558.15  4967.6    1556
  4976.1 1552.42  4985.9 1551.42  4986.4 1550.92  4995.6 1551.42  5007.8 1551.52
  5018.4 1553.19  5032.6    1559  5055.1 1560.74  5188.1 1557.45  5258.8 1560.69
  5287.1 1564.26  5329.5  1572.3    5372 1583.43  5414.4 1590.21    5570 1627.47
#Mann= 6 ,-1 , 0
  4246.5    .035       0  4740.8     .12       0  4799.9    .035       0
  4985.9    .035       0  4995.6    .035       0  5055.1     .12       0
Bank Sta=4985.9,4995.6
XS Rating Curve= 0 ,0
Exp/Cntr=0.3,0.1

Type RM Length L Ch R = 1 ,34239   ,1512,1512,1512
BEGIN DESCRIPTION:
LITTLE JOSHUA CREEK 67.0
END DESCRIPTION:
XS GIS Cut Line= 3
      2020773.07      13867725.4      2021128.96       13867261.
      2021484.88     13866540.49
#Sta/Elev= 30
  4427.8 1604.11  4528.7 1594.27  4703.8 1579.65  4885.6 1565.15  4929.2 1555.45
    4946 1554.41  4964.5 1553.88  4980.4 1549.17  4980.9 1548.67  4990.2 1549.17
  5012.9 1551.04  5042.6  1557.9  5061.2 1558.55  5062.1 1558.45  5169.3 1558.07
  5401.7 1553.35  5558.8 1555.29  5575.7 1562.88  5581.3 1561.03  5598.1 1573.01
  5603.7 1570.86  5620.6 1585.23  5624.9 1583.75    5643 1597.24  5648.6 1595.29
  5655.3 1601.91  5677.6 1612.09  5715.9 1619.84  5732.8 1619.49  5816.5 1637.55
#Mann= 9 ,-1 , 0
  4427.8    .035       0  4528.7     .07       0  4703.8     .12       0
    4946     .07       0  4980.4     .05       0  4990.2     .07       0
  5061.2    .035       0  5062.1     .07       0  5169.3     .12       0
Bank Sta=4980.4,4990.2
XS Rating Curve= 0 ,0
Exp/Cntr=0.3,0.1

Type RM Length L Ch R = 1 ,32727   ,473,473,473
BEGIN DESCRIPTION:
LITTLE JOSHUA CREEK 66.0
END DESCRIPTION:
XS GIS Cut Line= 3
      2021025.01     13867874.99        2021825.       13867075.
      2022209.68     13866926.81
#Sta/Elev= 30
  3867.7 1584.69  3938.4 1578.34  4136.4 1565.86  4221.2    1565    4292 1559.95
  4534.1 1552.48  4574.8  1551.9  4603.1 1549.66  4631.4  1550.8  4702.5 1545.74
  4781.9 1544.05  4782.4 1543.55  4791.9 1544.05  4884.4 1547.39  4909.4 1547.61
  4942.5 1545.81  4970.8    1547  4995.5 1544.11  5052.6 1545.03  5068.7 1550.11
  5074.1 1556.33  5093.3 1566.76  5183.2 1573.93  5287.1 1578.35  5322.4 1581.97
  5347.1 1587.03    5377 1599.75  5384.8 1604.61  5401.7 1610.01  5411.3 1610.24
#Mann= 7 ,-1 , 0
  3867.7    .035       0  4534.1     .07       0  4702.5     .12       0
  4781.9     .05       0  4791.9     .12       0  4884.4    .033       0
  4909.4     .12       0
Bank Sta=4781.9,4791.9
XS Rating Curve= 0 ,0
Exp/Cntr=0.3,0.1

Type RM Length L Ch R = 1 ,32254   ,458,458,458
BEGIN DESCRIPTION:
LITTLE JOSHUA CREEK 65.0
END DESCRIPTION:
XS GIS Cut Line= 3
      2021541.29       13868307.        2021725.       13867475.
      2021975.01       13867325.
#Sta/Elev= 30
  4148.3 1584.72  4160.6 1584.07  4187.4 1577.16  4231.1 1573.67  4293.7 1570.55
  4437.1 1566.81  4672.6 1562.29  4682.9 1561.51  4698.6 1556.59  4703.7 1556.85
  4742.2 1551.59  4747.3 1551.87  4764.8 1548.71    4791 1546.15  4796.1 1546.54
  4826.2 1544.23  4843.6  1544.2  4943.6 1544.49  5008.9 1543.97  5009.4 1543.47
  5018.9 1543.97  5103.4 1548.35    5117 1550.83  5128.1 1551.72  5151.9 1553.83
    5183 1560.44    5220 1564.15  5241.4 1567.54  5278.3 1570.85  5291.9 1573.04
#Mann= 6 ,-1 , 0
  4148.3    .035       0  4843.6     .07       0  4943.6     .12       0
  5008.9     .05       0  5018.9     .12       0  5128.1     .12       0
Bank Sta=5008.9,5018.9
XS Rating Curve= 0 ,0
Exp/Cntr=0.3,0.1

Type RM Length L Ch R = 1 ,31796   ,479,479,479
BEGIN DESCRIPTION:
LITTLE JOSHUA CREEK 64.0
END DESCRIPTION:
XS GIS Cut Line= 3
      2021610.75     13868354.73        2022075.       13867675.
        2022025.       13867325.
#Sta/Elev= 30
  4171.7 1581.16  4188.8 1580.44  4203.7 1581.51  4209.8 1580.08  4218.7 1581.21
  4224.7 1579.42  4239.6 1579.15  4347.3 1569.87    4618 1562.88  4742.8 1561.54
    4814 1562.37  4879.7 1560.19  4894.6 1557.03  4900.7 1557.68  4909.5 1553.78
  4915.6  1553.4  4919.6 1550.92  4930.5 1545.89  4946.4 1544.05  4946.9 1543.55
  4956.5 1544.05  5059.5 1544.07  5156.5 1544.62  5166.6  1545.9  5186.8 1551.62
    5207 1553.94  5267.6 1565.58  5297.9 1575.84  5318.1 1578.76  5348.4 1580.21
#Mann= 7 ,-1 , 0
  4171.7    .035       0    4618     .07       0  4742.8    .035       0
  4919.6     .07       0  4946.4     .05       0  4956.5     .07       0
  5059.5     .12       0
Bank Sta=4946.4,4956.5
XS Rating Curve= 0 ,0
Exp/Cntr=0.3,0.1

Type RM Length L Ch R = 1 ,31683   ,366,366,366
BEGIN DESCRIPTION:
LITTLE JOSHUA CREEK 63.5
END DESCRIPTION:
XS GIS Cut Line= 4
      2021886.58     13868506.39      2022169.26     13867827.22
      2022174.47     13867636.55        2022068.     13867299.03
#Sta/Elev= 30
  4156.1  1567.7  4571.5 1558.97    4637 1557.14  4689.6 1554.78  4790.4 1553.79
    4914 1558.07    4919 1557.65    4924 1554.84    4964 1544.12    4979 1543.95
  4979.5 1543.45  4989.1 1543.95    5024 1544.08    5054  1551.2  5075.9 1554.37
  5125.7  1555.5  5130.9 1553.66  5157.5 1555.32  5195.6 1553.78  5200.9 1554.97
  5241.4 1554.95  5251.9 1554.52  5260.3 1552.52  5265.6 1554.59  5297.9 1554.73
  5330.3  1563.8  5335.8 1566.73  5367.9 1574.28  5409.2 1580.87  5436.4 1582.72
#Mann= 6 ,-1 , 0
  4156.1    .035       0  4571.5     .07       0    4637    .035       0
    4979    .035       0  4989.1    .035       0  5075.9     .12       0
Bank Sta=4979,4989.1
XS Rating Curve= 0 ,0
Exp/Cntr=0.3,0.1

Type RM Length L Ch R = 1 ,31317   ,460,460,460
BEGIN DESCRIPTION:
LITTLE JOSHUA CREEK 63.0
END DESCRIPTION:
XS GIS Cut Line= 3
       2022490.9     13868376.43      2022465.03     13867685.71
        2022275.     13867325.01
#Sta/Elev= 30
  4308.8 1569.31  4550.4 1558.04  4620.4 1553.14  4660.5 1551.37  4670.5  1552.3
  4690.5 1549.37  4698.7 1549.69  4819.4 1544.93  4860.6 1542.35  4922.2 1535.04
  4930.7 1535.37  4960.7 1528.95  4980.7 1528.03  4997.9 1537.58  5036.3 1540.29
  5078.5 1540.33  5096.7 1539.33  5125.1 1531.18  5164.8 1523.93  5165.3 1523.43
  5175.9 1523.93    5193 1528.82  5206.9 1530.57  5223.3 1536.79  5245.3 1541.73
  5283.4  1546.7  5289.4 1548.92  5311.4 1550.04  5354.1 1557.69  5407.7 1573.56
#Mann= 7 ,-1 , 0
  4308.8    .035       0  4698.7     .07       0  4819.4     .12       0
  4922.2     .07       0  5078.5     .12       0  5164.8     .05       0
  5175.9     .12       0
Bank Sta=5164.8,5175.9
XS Rating Curve= 0 ,0
Exp/Cntr=0.3,0.1

Type RM Length L Ch R = 1 ,30857   ,347,347,347
BEGIN DESCRIPTION:
LITTLE JOSHUA CREEK 62.0
END DESCRIPTION:
XS GIS Cut Line= 3
      2022652.39     13868285.35      2022839.03     13867517.08
      2022782.73     13867018.97
#Sta/Elev= 30
  4216.4 1564.35  4329.1 1558.02  4415.3 1548.48  4597.5 1540.49  4626.6 1542.05
  4638.7 1538.49  4673.5 1544.35  4741.6 1538.42  4932.7 1533.58  4947.4 1534.84
  4957.7 1531.75  4965.8 1521.26  4971.1 1521.69  4993.3 1519.34  4993.8 1518.84
  5004.5 1519.34  5029.2 1520.12  5059.4 1533.21    5086 1550.84  5170.1 1565.34
  5260.6 1574.27  5265.6 1569.82  5294.7 1566.34    5311 1566.02  5341.2 1580.96
  5350.4 1583.69  5355.4 1580.94  5431.8 1607.81  5482.1 1615.23  5508.3 1623.17
#Mann= 7 ,-1 , 0
  4216.4    .035       0  4415.3     .07       0  4932.7    .035       0
  4971.1     .07       0  4993.3     .05       0  5004.5     .07       0
  5294.7     .12       0
Bank Sta=4993.3,5004.5
XS Rating Curve= 0 ,0
Exp/Cntr=0.3,0.1

Type RM Length L Ch R = 1 ,30510   ,470,470,470
BEGIN DESCRIPTION:
LITTLE JOSHUA CREEK 61.0
END DESCRIPTION:
XS GIS Cut Line= 3
      2022782.63     13868398.12        2023125.       13867675.
      2023138.51     13867200.27
#Sta/Elev= 30
  4199.9  1573.8  4377.8  1560.4  4383.3 1563.45  4400.5 1559.15  4451.6 1558.06
  4457.8 1554.14    4480 1550.39  4680.6 1536.41  4752.8 1534.23  4775.6 1537.65
  4781.1 1543.34  4798.3 1533.78  4825.3  1532.3  4843.8 1532.23  4856.1 1536.24
  4894.8 1528.53  4963.3 1524.48  5004.4 1518.57  5004.9 1518.07  5015.6 1518.57
    5040 1518.91    5080    1526    5100 1537.31    5110 1548.59    5120 1554.79
  5137.5 1561.44  5175.4  1564.9  5180.4 1562.16    5194 1563.03  5474.9 1596.88
#Mann= 8 ,-1 , 0
  4199.9    .035       0  4680.6     .07       0  4825.3    .035       0
  4963.3     .07       0  5004.4     .05       0  5015.6     .07       0
  5137.5     .12       0    5194     .07       0
Bank Sta=5004.4,5015.6
XS Rating Curve= 0 ,0
Exp/Cntr=0.3,0.1

Type RM Length L Ch R = 1 ,30040   ,348,348,348
BEGIN DESCRIPTION:
LITTLE JOSHUA CREEK 60.0
END DESCRIPTION:
XS GIS Cut Line= 3
        2023225.       13868225.        2023425.       13868025.
      2023437.99     13867261.05
#Sta/Elev= 30
  4716.8 1548.13  4719.5 1548.13  4759.2 1545.71  4773.4 1543.31  4815.8 1531.13
  4844.1 1527.01  4858.3 1526.42  4914.8 1523.65  4971.4  1516.5    5004 1516.26
  5004.5 1515.76  5015.2 1516.26  5049.6 1520.15  5059.7 1522.26  5077.1 1520.97
  5109.7 1522.69  5129.7 1526.48  5159.7 1529.82  5201.4 1532.76  5268.4 1536.22
  5294.2 1537.95  5319.7 1541.63  5339.7  1541.6  5369.7 1544.55  5459.7  1559.3
  5499.7  1561.2  5699.7 1579.12  5739.7 1584.33  5759.3 1590.11  5763.7 1590.11
#Mann= 8 ,-1 , 0
  4716.8    .035       0  4719.5     .12       0  4858.3    .035       0
    5004    .035       0  5015.2    .035       0  5077.1     .07       0
  5201.4    .035       0  5268.4     .07       0
Bank Sta=5004,5015.2
XS Rating Curve= 0 ,0
Exp/Cntr=0.3,0.1

Type RM Length L Ch R = 1 ,29692   ,684,684,684
BEGIN DESCRIPTION:
LITTLE JOSHUA CREEK 59.0
END DESCRIPTION:
XS GIS Cut Line= 3
      2023142.82     13868567.45      2023637.64     13868168.12
      2023589.95      13867235.9
#Sta/Elev= 30
  4380.8 1564.29  4420.1 1562.79  4440.9 1568.81  4447.8  1568.7  4461.7 1567.33
  4484.1 1558.82  4504.9 1555.86  4639.8  1547.6    4668 1546.37  4704.8 1537.22
  4711.2 1537.07  4725.6  1531.8  4771.5 1523.31  4810.4 1522.68  4824.8  1519.8
  4874.3 1515.94  4940.4 1516.04  5009.5 1515.92    5010 1515.42  5020.8 1515.92
  5049.8 1521.28  5119.9 1526.25  5326.5 1530.77  5332.3    1531  5500.4 1540.96
  5640.6 1556.39  5740.7 1565.03  5780.8 1571.32  5910.9 1580.35  5950.1 1586.41
#Mann= 8 ,-1 , 0
  4380.8    .035       0  4639.8     .12       0  4771.5    .035       0
  4940.4     .07       0  5009.5     .05       0  5020.8     .07       0
  5326.5    .035       0  5332.3     .07       0
Bank Sta=5009.5,5020.8
XS Rating Curve= 0 ,0
Exp/Cntr=0.3,0.1

Type RM Length L Ch R = 1 ,29008   ,251,251,251
BEGIN DESCRIPTION:
LITTLE JOSHUA CREEK 58.0
END DESCRIPTION:
XS GIS Cut Line= 3
      2023303.46      13868888.6      2024080.35     13868376.46
      2024324.97     13868125.03
#Sta/Elev= 30
  4064.3 1562.01  4233.8 1549.88  4298.8  1548.1  4313.9 1551.09  4319.9 1549.31
    4329 1552.86    4335 1549.17  4341.6 1553.43    4350 1553.44  4365.1 1548.65
  4392.2 1543.43  4407.2 1542.37  4627.7 1536.52  4742.2 1534.98  4768.6 1531.64
  4783.7 1527.78  4810.7 1517.19  4902.7 1516.17  5000.2 1515.86  5000.7 1515.36
  5012.3 1515.86  5083.9 1521.31  5127.3 1521.87  5197.1 1526.18  5232.6 1531.27
  5260.9  1539.6    5282 1550.29  5286.7 1551.24  5310.3 1558.93  5345.6 1563.14
#Mann= 8 ,-1 , 0
  4064.3    .035       0  4627.7     .07       0  4742.2    .035       0
  4902.7    .033       0  5000.2    .033       0  5012.3    .033       0
  5127.3     .07       0  5286.7     .12       0
Bank Sta=5000.2,5012.3
XS Rating Curve= 0 ,0
Exp/Cntr=0.3,0.1

Type RM Length L Ch R = 1 ,28757   ,86,86,86
BEGIN DESCRIPTION:
LITTLE JOSHUA CREEK 57.0
END DESCRIPTION:
XS GIS Cut Line= 3
      2023446.67     13869088.26        2024275.       13868525.
      2024407.45     13868172.88
#Sta/Elev= 30
  3998.6 1553.97  4133.5 1548.65  4201.8 1547.26  4403.1 1540.53  4424.1 1541.45
  4468.2 1538.35  4504.5 1538.34  4561.7 1535.26  4576.7 1536.27  4589.1 1534.59
  4631.3 1533.78  4680.3 1532.71  4705.4 1532.13  4726.4 1533.87  4806.8 1529.32
  4843.1 1521.21  4885.1 1516.22    5044 1516.13  5069.8 1516.01  5070.3 1515.51
  5081.9 1516.01  5127.6 1518.29  5180.7 1519.26  5192.6 1520.74  5235.3 1533.25
  5256.7 1537.29  5271.4 1542.53  5278.1  1546.7  5331.9 1562.35  5376.5  1566.6
#Mann= 9 ,-1 , 0
  3998.6     .07       0  4133.5     .12       0  4201.8    .035       0
  4631.3     .07       0  4680.3    .035       0    5044    .033       0
  5069.8    .035       0  5081.9    .033       0  5127.6     .12       0
Bank Sta=5069.8,5081.9
XS Rating Curve= 0 ,0
Exp/Cntr=0.3,0.1

Type RM Length L Ch R = 1 ,28671   ,358,358,358
BEGIN DESCRIPTION:
LITTLE JOSHUA CREEK 56.5
END DESCRIPTION:
XS GIS Cut Line= 3
      2024255.72     13868879.97       2024342.1       13868575.
      2024474.91      13868218.5
#Sta/Elev= 30
  4682.8 1528.92    4701 1530.03    4714 1529.26  4760.7  1526.6  4768.9 1523.54
  4774.1 1524.98  4781.5 1522.03  4802.3 1519.81  4813.2 1517.43  4841.1  1515.1
  4841.6  1514.6  4853.2  1515.1  4854.3    1516    4875 1516.24  4903.5 1518.67
    4915    1520  4920.2 1523.26    4927  1524.8  5081.2 1526.71  5181.2 1526.39
  5220.7 1528.23  5245.2  1534.5    5276 1544.69  5287.9 1551.31  5306.4 1555.29
  5311.7 1559.13  5336.7 1560.77    5342 1562.94  5361.7 1564.65  5380.2 1568.94
#Mann= 6 ,-1 , 0
  4682.8     .07       0    4714    .035       0  4841.1     .05       0
  4853.2    .035       0  4903.5     .07       0  5081.2     .12       0
Bank Sta=4841.1,4853.2
XS Rating Curve= 0 ,0
Exp/Cntr=0.3,0.1

Type RM Length L Ch R = 1 ,28313   ,468,468,468
BEGIN DESCRIPTION:
LITTLE JOSHUA CREEK 56.0
END DESCRIPTION:
XS GIS Cut Line= 3
      2024258.22     13869338.74        2024625.       13868725.
      2024897.69     13868252.99
#Sta/Elev= 30
  4276.4 1544.22  4304.6 1543.12    4341 1536.94  4421.4 1533.52  4493.8 1525.15
  4569.2 1515.23  4590.6 1516.21  4618.6 1512.77  4639.9 1514.62  4707.4 1517.87
    4791 1516.24  4842.6 1514.22  4890.2 1511.79  4925.2 1511.48  4940.8  1502.8
  4982.4 1498.45  4982.9 1497.95  4994.5 1498.45  5049.1 1498.56    5086  1502.8
  5160.1 1520.96  5203.2 1525.99  5233.9 1535.87  5268.6 1552.22  5350.7 1565.62
  5460.1 1588.87  5475.9 1593.68  5481.7  1598.4  5497.5    1600  5536.5 1611.02
#Mann= 11 ,-1 , 0
  4276.4     .07       0    4341     .12       0  4493.8     .07       0
  4639.9     .12       0    4791    .035       0  4842.6     .12       0
  4890.2     .07       0  4982.4     .05       0  4994.5     .07       0
    5086     .12       0  5350.7     .07       0
Bank Sta=4982.4,4994.5
XS Rating Curve= 0 ,0
Exp/Cntr=0.3,0.1

Type RM Length L Ch R = 1 ,27845   ,434,434,434
BEGIN DESCRIPTION:
LITTLE JOSHUA CREEK 55.0
END DESCRIPTION:
XS GIS Cut Line= 3
      2024206.24     13869509.26        2025025.       13868925.
        2025025.     13868625.05
#Sta/Elev= 30
  3993.5 1551.11  4208.3 1544.13  4238.5 1543.05  4247.1 1541.82  4253.3 1539.09
  4274.2 1537.21  4347.9 1533.29  4383.6 1529.52    4434 1515.44  4454.9 1511.88
  4532.9 1509.13  4655.4 1508.59  4677.3  1506.6  4695.1  1508.6  4769.5 1510.58
  4855.5 1507.02  4870.2 1505.33    4885 1499.98  4914.9 1499.31  4985.9 1498.23
  4986.4 1497.73  4998.1 1498.23  5039.3 1502.87  5059.3 1506.88  5077.1 1513.77
  5112.3 1520.72  5169.3 1537.08  5239.3 1552.91  5269.3 1561.18  5299.3 1566.61
#Mann= 11 ,-1 , 0
  3993.5    .035       0  4208.3     .07       0  4274.2     .12       0
  4532.9     .07       0  4695.1     .12       0  4769.5     .07       0
  4914.9     .12       0  4985.9     .05       0  4998.1     .12       0
  5077.1     .07       0  5112.3     .12       0
Bank Sta=4985.9,4998.1
XS Rating Curve= 0 ,0
Exp/Cntr=0.3,0.1

Type RM Length L Ch R = 1 ,27411   ,470,470,470
BEGIN DESCRIPTION:
LITTLE JOSHUA CREEK 54.0
END DESCRIPTION:
XS GIS Cut Line= 3
      2024361.51     13869502.15        2025125.       13869325.
      2025267.92     13869180.38
#Sta/Elev= 30
  4216.1 1548.52  4240.2 1546.83  4286.7 1545.81  4388.6 1542.95    4401 1543.03
  4455.8 1532.07  4491.4 1528.28  4527.7  1526.4  4568.7 1520.99  4599.5 1510.18
  4630.3 1502.05  4661.1 1498.54  4667.1 1500.09  4681.6 1500.74  4784.3 1502.34
  4800.2 1501.52  4805.4  1502.8    4848 1501.38  4876.7 1498.61  4919.1 1498.51
  4921.9  1498.5  4922.4    1498  4934.1  1498.5    4976 1498.61  4989.6 1499.89
  4997.3 1502.87  5021.1 1503.63  5060.3 1507.51    5119 1510.95  5203.2 1514.16
#Mann= 8 ,-1 , 0
  4216.1    .035       0  4286.7     .07       0  4388.6     .12       0
  4919.1    .033       0  4921.9    .033       0  4934.1    .033       0
  5060.3     .12       0    5119    .035       0
Bank Sta=4921.9,4934.1
XS Rating Curve= 0 ,0
Exp/Cntr=0.3,0.1

Type RM Length L Ch R = 1 ,26941   ,420,420,420
BEGIN DESCRIPTION:
LITTLE JOSHUA CREEK 53.0
END DESCRIPTION:
XS GIS Cut Line= 3
      2025224.99     13869974.95        2025125.       13869625.
      2025375.02     13869024.96
#Sta/Elev= 30
    4636 1547.34  4677.6    1544  4689.9 1541.09  4698.4 1537.97  4725.7 1530.83
  4764.7 1526.82  4798.5 1517.54  4803.7 1518.23  4823.2 1514.29  4832.3 1511.46
  4837.5 1510.92    4844 1507.22  4864.8 1500.08  4871.3 1499.09  5008.1 1498.31
  5008.6 1497.81    5021 1498.31  5040.9 1498.69  5120.7 1498.74  5139.2 1499.91
  5144.6 1501.72  5173.8 1504.14  5251.1 1505.54  5337.6 1508.35  5380.7 1509.87
  5399.2 1511.73  5411.6 1511.12  5452.2 1513.47  5481.5  1513.9    5650 1524.91
#Mann= 7 ,-1 , 0
    4636    .035       0  4689.9     .07       0  5008.1     .05       0
    5021     .07       0  5040.9    .033       0  5251.1     .07       0
  5337.6    .035       0
Bank Sta=5008.1,5021
XS Rating Curve= 0 ,0
Exp/Cntr=0.3,0.1

Type RM Length L Ch R = 1 ,26521   ,746,746,746
BEGIN DESCRIPTION:
LITTLE JOSHUA CREEK 52.0
END DESCRIPTION:
XS GIS Cut Line= 3
       2025514.4     13869864.57        2025475.       13869575.
      2025389.68     13869154.71
#Sta/Elev= 30
  4703.4 1531.73  4723.1 1528.84  4753.4 1525.87  4763.5    1524  4793.8 1515.95
  4809.6 1510.82  4814.6 1510.67  4848.8 1505.64  4864.4 1504.94  4914.9 1506.75
    4925 1505.12  4935.1 1500.28  4945.2 1498.67  4965.4 1499.08  4999.6 1498.45
  5009.4  1498.3  5009.9  1497.8  5021.9  1497.8  5022.4  1498.3  5055.2 1498.59
  5148.7 1498.38  5167.8 1500.19  5188.6 1500.43  5221.9 1500.76  5240.5 1501.57
  5260.9 1503.24  5274.2 1505.09    5312 1507.08  5358.3 1510.67  5424.5 1515.59
#Mann= 9 ,-1 , 0
  4703.4    .035       0  4848.8     .07       0  4999.6    .033       0
  5009.4    .033       0  5022.4    .033       0  5055.2     .07       0
  5188.6    .035       0  5221.9     .07       0  5358.3     .12       0
Bank Sta=5009.4,5022.4
XS Rating Curve= 0 ,0
Exp/Cntr=0.3,0.1

Type RM Length L Ch R = 1 ,25775   ,41,41,41
BEGIN DESCRIPTION:
LITTLE JOSHUA CREEK 51.0
END DESCRIPTION:
XS GIS Cut Line= 3
      2026052.21     13869584.64      2025894.85      13869054.4
      2025624.98     13868474.96
#Sta/Elev= 30
  4446.9 1513.02  4486.4 1511.79  4541.2 1502.25  4563.3 1499.32  4726.9 1498.54
  4863.8 1499.37  4971.1 1498.21  4971.6 1497.71  4984.1 1498.21  5018.2 1498.29
  5043.5 1498.39  5076.6 1502.61  5098.6 1506.02  5128.3 1513.22  5158.4 1516.71
  5202.2 1520.37  5208.9 1522.85  5238.4 1527.01  5286.2 1537.21  5330.3 1552.32
  5362.3 1555.44  5407.5 1563.44  5429.6  1568.2    5442 1572.59  5464.8 1576.84
  5510.6 1581.72  5550.8  1590.9  5579.2 1602.38  5607.6 1605.15  5639.2  1612.4
#Mann= 9 ,-1 , 0
  4446.9    .035       0  4541.2     .07       0  4726.9    .033       0
  4971.1    .033       0  4984.1    .033       0  5018.2     .12       0
  5128.3     .07       0  5158.4    .035       0  5238.4     .07       0
Bank Sta=4971.1,4984.1
XS Rating Curve= 0 ,0
Exp/Cntr=0.3,0.1

Type RM Length L Ch R = 1 ,25734   ,569,569,569
BEGIN DESCRIPTION:
LITTLE JOSHUA CREEK 50.5
END DESCRIPTION:
XS GIS Cut Line= 4
      2026128.27      13869571.6       2025958.7     13869125.31
        2025925.       13869025.      2025711.59     13868572.88
#Sta/Elev= 30
  4420.3 1512.72  4457.4 1512.03  4486.2 1510.64  4583.4 1500.96  4588.8 1503.46
  4638.3    1501  4643.7 1503.93    4652 1503.89  4668.4 1500.21  4673.8 1504.07
  4693.2 1502.18  4698.6 1504.56  4723.3 1502.58  4728.7 1504.59  4788.6  1504.5
  4876.7 1503.78  4949.8 1498.07  4950.3 1497.57  4962.8 1498.07  4988.5 1498.46
  5040.5 1499.76  5098.1 1507.07  5209.9 1523.89  5217.3 1524.95  5268.2 1533.09
  5313.2 1546.29  5324.8    1552  5387.6 1558.25  5461.4 1572.32  5503.5 1577.95
#Mann= 10 ,-1 , 0
  4420.3     .07       0  4457.4    .035       0  4486.2     .07       0
  4788.6    .033       0  4949.8     .05       0  4962.8    .033       0
  4988.5     .12       0  5098.1     .07       0  5209.9    .035       0
  5217.3     .07       0
Bank Sta=4949.8,4962.8
XS Rating Curve= 0 ,0
Exp/Cntr=0.3,0.1
