HEC-RAS study CURRY CREEK.prj: CURRY CREEK Base Level Engineering

--- CURRY CREEK.g01 (geometry) --- (continued)

Type RM Length L Ch R = 1 ,84537   ,509,509,509
BEGIN DESCRIPTION:
CURRY CREEK 136.0
END DESCRIPTION:
XS GIS Cut Line= 3
      2090561.94     13907454.34      2089673.01      13906982.1
       2088863.4     13906588.05
#Sta/Elev= 30
  3995.8 1457.65  4193.7 1451.67  4305.9 1443.79    4332 1439.27  4431.8 1432.72
  4541.6 1429.37  4649.6 1426.64  4745.6 1421.32  4775.9  1420.2  4792.2 1416.26
  4797.8 1417.27  4814.2 1414.41    4892 1413.28  4989.7 1401.81  4990.2 1401.31
  5007.1 1401.81    5029 1413.13  5051.6 1414.95  5223.3 1416.68  5400.9 1416.76
  5499.5 1419.48  5634.1 1425.42  5665.9    1433  5705.7 1446.34  5739.1 1455.81
  5745.3 1460.57  5767.6 1468.14  5806.7 1477.34  5879.9 1485.54  5902.8  1485.9
#Mann= 11 ,-1 , 0
  3995.8     .07       0  4305.9     .12       0  4431.8     .07       0
  4541.6     .12       0  4745.6     .07       0    4892     .12       0
  4989.7     .05       0  5007.1     .12       0  5223.3     .07       0
  5499.5     .12       0  5705.7     .07       0
Bank Sta=4989.7,5007.1
XS Rating Curve= 0 ,0
Exp/Cntr=0.3,0.1

Type RM Length L Ch R = 1 ,84028   ,481,481,481
BEGIN DESCRIPTION:
CURRY CREEK 135.0
END DESCRIPTION:
XS GIS Cut Line= 3
      2090600.01     13907350.01        2089675.       13906475.
      2089074.95     13906274.98
#Sta/Elev= 30
  3726.3 1456.08  3839.5 1452.45  4041.8 1441.51  4143.8 1436.52  4292.3 1431.84
  4313.3 1431.25  4320.6 1433.58  4341.6 1430.26  4386.7 1429.52  4479.7 1425.68
    4560 1423.13  4589.2 1421.15  4801.6 1417.61  4907.6 1413.54    4929 1407.59
  4964.2 1403.68  4969.7 1399.09  4970.2 1398.59  4987.1 1399.09  4992.5 1400.61
  4996.2 1405.11  5031.2 1408.51  5052.3 1413.79  5290.9 1413.31    5358 1415.05
  5401.2  1417.9  5431.8 1424.85  5537.2 1468.57    5611 1479.67  5632.1  1481.3
#Mann= 10 ,-1 , 0
  3726.3     .07       0  3839.5     .12       0  4041.8     .07       0
  4386.7     .12       0  4479.7     .07       0    4560     .12       0
  4969.7     .05       0  4987.1     .12       0  5290.9     .07       0
  5401.2     .12       0
Bank Sta=4969.7,4987.1
XS Rating Curve= 0 ,0
Exp/Cntr=0.3,0.1

Type RM Length L Ch R = 1 ,83547   ,483,483,483
BEGIN DESCRIPTION:
CURRY CREEK 134.0
END DESCRIPTION:
XS GIS Cut Line= 3
      2090550.02     13907100.03        2089775.       13906025.
      2089174.96       13906075.
#Sta/Elev= 30
  3675.4 1447.32  3983.4 1435.95  4119.6 1433.61  4149.1 1430.13  4218.3 1427.84
  4279.6 1425.43  4441.2 1419.88  4489.7 1418.54  4613.7 1416.79  4737.7  1416.6
  4764.5 1416.18  4901.3  1413.3    4943  1405.9  4987.2 1402.26  4993.3 1399.45
  5000.7 1398.92    5002 1396.78  5002.5 1396.28  5019.4 1396.78  5030.8 1402.62
  5063.4 1406.47    5081 1410.59  5252.4 1411.53  5351.6 1412.59  5424.6 1414.44
  5462.3 1417.74  5492.4 1426.86    5540 1449.82  5545.1 1449.94  5602.8 1466.65
#Mann= 12 ,-1 , 0
  3675.4     .12       0  4218.3     .07       0  4279.6    .035       0
  4441.2     .12       0  4489.7    .035       0  4613.7     .07       0
  4737.7    .035       0  4764.5     .12       0    5002     .05       0
  5019.4     .12       0  5252.4     .07       0  5351.6     .12       0
Bank Sta=5002,5019.4
XS Rating Curve= 0 ,0
Exp/Cntr=0.3,0.1

Type RM Length L Ch R = 1 ,83064   ,465,465,465
BEGIN DESCRIPTION:
CURRY CREEK 133.0
END DESCRIPTION:
XS GIS Cut Line= 3
      2090304.96     13906124.47        2089875.       13905575.
        2089475.       13905225.
#Sta/Elev= 30
  4302.3 1418.26  4325.8 1417.99  4755.7 1412.04    4779 1411.39  4909.6 1407.13
  4928.6 1404.04  4957.5 1402.85  4986.4 1396.66    4988  1395.1  4988.5  1394.6
  5005.7  1395.1  5007.1 1398.85  5013.8 1400.64    5028 1401.89  5049.8 1406.88
  5180.1 1408.58  5197.1  1408.9  5254.8 1410.39  5354.5 1420.43  5389.6 1431.98
  5397.2 1433.59  5411.4 1439.53    5439 1458.26  5453.2  1466.7    5475 1474.63
  5481.7 1478.34  5495.9 1483.27  5524.4 1485.32  5528.2 1486.96  5531.5 1486.96
#Mann= 9 ,-1 , 0
  4302.3     .07       0  4325.8    .035       0  4755.7     .12       0
    4779    .035       0  4909.6     .12       0    4988     .05       0
  5005.7     .12       0  5180.1     .07       0  5197.1     .12       0
Bank Sta=4988,5005.7
XS Rating Curve= 0 ,0
Exp/Cntr=0.3,0.1

Type RM Length L Ch R = 1 ,82599   ,412,412,412
BEGIN DESCRIPTION:
CURRY CREEK 132.0
END DESCRIPTION:
XS GIS Cut Line= 3
      2090674.97     13905674.98        2090075.       13905175.
      2089875.03     13904925.03
#Sta/Elev= 30
  4218.8 1420.33  4232.4 1420.72  4275.4 1417.42  4339.8  1414.7  4445.9 1411.41
  4531.2 1407.66  4807.8 1403.91  4850.7 1406.02  4879.4 1405.79  4914.2  1403.5
  4978.3 1399.96  4986.1 1397.01  4987.6 1393.08  4988.1 1392.58  5005.4 1393.08
  5021.4 1399.02  5027.8 1399.78  5042.2  1404.5  5106.2 1405.13  5127.8 1407.33
  5149.5 1411.16  5163.9 1415.65  5205.5 1435.34  5242.3 1447.03  5255.9 1452.86
  5276.7 1457.49  5283.9 1460.28  5306.3 1463.23  5312.7 1465.42  5319.9 1466.21
#Mann= 6 ,-1 , 0
  4218.8     .12       0  4339.8    .035       0  4914.2     .12       0
  4987.6     .05       0  5005.4     .12       0  5276.7     .07       0
Bank Sta=4987.6,5005.4
XS Rating Curve= 0 ,0
Exp/Cntr=0.3,0.1

Type RM Length L Ch R = 1 ,82187   ,446,446,446
BEGIN DESCRIPTION:
CURRY CREEK 131.0
END DESCRIPTION:
XS GIS Cut Line= 3
      2090925.01     13905475.01        2090325.       13904875.
      2089875.02     13904775.01
#Sta/Elev= 30
  4146.8 1426.06  4232.3 1421.12  4288.2 1415.74    4359 1411.39  4503.2 1406.76
  4754.9 1402.16  4853.9 1401.97  4924.6 1403.78  4947.8 1401.28  4981.2 1398.05
  4982.9 1391.24  4983.4 1390.74  5000.7 1391.24  5014.6 1393.03  5026.1  1398.6
  5068.3 1402.47  5138.8 1402.16  5179.7 1404.67  5204.1 1408.27  5247.6 1422.43
  5252.7 1422.51  5291.1 1435.35  5296.3 1435.15  5302.7 1438.71  5339.8 1450.19
  5353.9 1453.27  5388.5 1464.42  5405.1 1470.98  5431.8 1474.27  5456.3 1477.38
#Mann= 7 ,-1 , 0
  4146.8     .12       0  4232.3    .035       0  4503.2     .07       0
  4947.8     .12       0  4982.9     .05       0  5000.7     .12       0
  5431.8     .07       0
Bank Sta=4982.9,5000.7
XS Rating Curve= 0 ,0
Exp/Cntr=0.3,0.1

Type RM Length L Ch R = 1 ,81930   ,1013,1013,1013
BEGIN DESCRIPTION:
CURRY CREEK 130.0
END DESCRIPTION:
XS GIS Cut Line= 3
       2090959.1     13905223.48      2090483.29     13904686.12
      2090075.01     13904325.01
#Sta/Elev= 30
  4268.3 1420.54  4291.7 1420.14  4312.7 1417.59    4317 1417.27    4452 1407.22
  4539.3 1403.73  4645.5 1402.55  4780.2 1401.73  4843.7 1403.18  4857.9 1402.62
  4865.5 1400.57  4879.7 1399.56  4964.2 1397.59  4983.4 1394.13  4983.8 1389.16
  4984.3 1388.66  5001.9 1389.16  5013.8 1396.21    5028 1397.31  5049.7 1401.61
  5091.5 1400.35  5141.8 1401.14  5290.6 1409.26  5332.4 1413.74  5354.2 1418.43
  5417.7 1442.17  5438.7 1450.58  5495.6 1469.29  5503.1 1470.88  5531.1 1472.03
#Mann= 7 ,-1 , 0
  4268.3     .12       0  4312.7    .035       0    4317     .12       0
    4452    .035       0  4983.8     .05       0  5001.9    .035       0
  5417.7    .035       0
Bank Sta=4983.8,5001.9
XS Rating Curve= 0 ,0
Exp/Cntr=0.3,0.1

Type RM Length L Ch R = 1 ,81329   ,446,446,446
BEGIN DESCRIPTION:
CURRY CREEK 129.0
END DESCRIPTION:
XS GIS Cut Line= 3
      2091175.02     13904575.02        2090875.       13904275.
      2090324.98     13904124.99
#Sta/Elev= 30
  4571.1  1408.1  4610.1 1405.69  4671.6 1397.92    4755 1395.96  4811.5 1397.92
  4938.8 1399.14    4953 1398.48  4967.1 1395.76  4991.9 1388.28  5008.8 1386.49
  5009.3 1385.99    5027 1386.49  5036.9 1393.62  5057.6 1397.86  5078.3 1399.19
  5111.9  1397.6  5161.2 1397.69    5231  1400.9  5293.6 1407.24    5315 1409.93
  5327.1  1413.3  5354.7 1412.93  5368.5 1418.92  5389.3 1422.16  5399.6 1427.29
  5434.2 1439.48  5461.8 1445.38  5482.6 1451.78    5524 1461.24  5565.5 1464.65
#Mann= 8 ,-1 , 0
  4571.1    .045       0  4610.1     .07       0  4671.6    .045       0
  5008.8    .045       0    5027    .045       0  5111.9     .07       0
    5231    .035       0  5293.6     .07       0
Bank Sta=5008.8,5027
XS Rating Curve= 0 ,0
Exp/Cntr=0.3,0.1

Type RM Length L Ch R = 1 ,80883   ,423,423,423
BEGIN DESCRIPTION:
CURRY CREEK 128.0
END DESCRIPTION:
XS GIS Cut Line= 3
      2091275.01     13904525.04        2091175.       13903975.
      2089971.61     13903742.51
#Sta/Elev= 30
  4441.2 1407.43  4457.4 1407.08  4609.2 1399.15  4725.8 1393.45  4916.9 1396.23
  4968.5 1393.64  4979.9 1389.47    4981 1385.15  4981.5 1384.65  4999.2 1385.15
  5020.6 1385.32    5041  1393.5    5078 1397.08    5153 1389.25  5186.7 1390.38
    5204 1396.16  5290.4 1398.95  5338.6 1407.66  5445.8 1424.44  5456.1 1429.09
    5479 1433.36  5540.1 1433.05  5606.4 1441.24  5698.1 1432.82    5710 1432.26
  5715.1 1427.76  5761.9 1426.59  5774.3 1421.94  5886.3 1419.76  6225.9 1433.04
#Mann= 9 ,-1 , 0
  4441.2    .035       0  4457.4     .07       0  4609.2    .045       0
  4916.9     .07       0    4981     .05       0  4999.2     .07       0
  5338.6    .035       0  5456.1     .07       0  5698.1    .035       0
Bank Sta=4981,4999.2
XS Rating Curve= 0 ,0
Exp/Cntr=0.3,0.1

Type RM Length L Ch R = 1 ,80460   ,421,421,421
BEGIN DESCRIPTION:
CURRY CREEK 127.0
END DESCRIPTION:
XS GIS Cut Line= 3
        2091475.     13904375.01        2091525.       13903775.
       2090629.5     13902730.52
#Sta/Elev= 30
  4397.9  1401.9  4427.7 1401.13  4701.5 1389.88  4946.6 1395.14  4969.9 1391.88
    4990 1381.03  4997.8 1380.27  4998.3 1379.77  5016.5 1380.27  5042.2 1391.76
    5086 1396.16  5134.4 1391.42  5193.9 1394.64  5389.1 1395.66  5418.7 1399.95
  5439.6  1395.8  5468.1 1396.69  5560.3 1415.05  5631.6 1424.12  5659.1 1423.29
  5673.3 1428.03    5681 1435.05  5714.3 1439.04  5723.8 1441.59  5730.4 1439.06
  5908.2 1471.65  6191.4 1506.39  6267.5  1526.2  6297.8 1537.83  6375.8 1540.99
#Mann= 9 ,-1 , 0
  4397.9     .07       0  4427.7    .045       0  4946.6     .07       0
  4997.8     .05       0  5016.5     .07       0    5086    .035       0
  5193.9     .07       0  5389.1     .12       0  5714.3     .07       0
Bank Sta=4997.8,5016.5
XS Rating Curve= 0 ,0
Exp/Cntr=0.3,0.1

Type RM Length L Ch R = 1 ,80039   ,447,447,447
BEGIN DESCRIPTION:
CURRY CREEK 126.0
END DESCRIPTION:
XS GIS Cut Line= 3
      2091674.99     13904575.04        2091875.       13903575.
        2091675.       13902975.
#Sta/Elev= 30
  3979.7 1407.92  4071.5 1404.63  4142.9 1398.91  4208.1 1396.84  4464.2 1391.84
  4642.6  1386.7  4731.8  1387.3  4831.5 1390.71  4877.2 1391.76  4897.6 1393.93
  4931.2 1392.25  4958.8 1383.18  4969.8 1377.11  4970.3 1376.61  4988.5 1377.11
  4989.4 1383.84    4997  1389.9  5010.1 1390.39  5020.6 1392.91  5032.5  1392.9
  5137.3 1389.93  5263.1 1389.38  5452.8 1395.47  5484.4 1394.29  5505.5 1398.11
    5520 1402.78  5547.7 1416.73  5558.2 1423.64  5589.8 1438.59    5632 1451.63
#Mann= 10 ,-1 , 0
  3979.7     .07       0  4208.1    .045       0  4731.8    .035       0
  4831.5    .045       0  4931.2    .035       0  4969.8    .035       0
  4988.5    .035       0  5032.5     .07       0  5137.3    .035       0
    5520     .12       0
Bank Sta=4969.8,4988.5
XS Rating Curve= 0 ,0
Exp/Cntr=0.3,0.1

Type RM Length L Ch R = 1 ,79592   ,469,469,469
BEGIN DESCRIPTION:
CURRY CREEK 125.0
END DESCRIPTION:
XS GIS Cut Line= 3
      2093077.84     13904804.21        2092225.       13903375.
      2091662.89     13902720.86
#Sta/Elev= 30
  3330.9 1414.85  3418.9 1409.45  3452.8 1406.04  3748.5 1388.24  3965.1 1383.18
  4001.2 1382.59  4081.8 1382.59  4184.1 1382.62  4198.5 1382.56  4315.2 1382.99
  4466.2  1382.6  4787.1 1388.33  4960.2 1392.15  4998.5 1386.44  4999.6 1373.47
  5000.1 1372.97  5018.3 1373.47  5051.7 1386.56  5117.2 1390.98  5248.2 1389.13
  5364.4 1389.62  5415.2 1394.52  5463.2 1405.51  5477.5 1416.82  5520.3 1434.97
  5555.4 1443.33    5584 1455.09  5626.7 1463.21  5710.1 1468.78  5857.7 1472.88
#Mann= 18 ,-1 , 0
  3330.9     .07       0  3418.9     .12       0  3452.8     .07       0
  3748.5    .035       0  3965.1     .07       0  4001.2    .035       0
  4081.8     .07       0  4184.1    .035       0  4198.5     .07       0
  4315.2    .035       0  4466.2    .045       0  4787.1    .035       0
  4999.6    .035       0  5018.3    .035       0  5117.2     .07       0
  5248.2    .035       0  5415.2     .12       0  5710.1     .07       0
Bank Sta=4999.6,5018.3
XS Rating Curve= 0 ,0
Exp/Cntr=0.3,0.1

Type RM Length L Ch R = 1 ,79123   ,478,478,478
BEGIN DESCRIPTION:
CURRY CREEK 124.0
END DESCRIPTION:
XS GIS Cut Line= 3
        2093225.     13904825.01        2092475.       13903025.
      2092274.97     13902974.99
#Sta/Elev= 30
  3048.6 1415.91  3050.3 1415.91  3233.3 1409.84  3286.2 1406.25  3376.3 1402.49
  3429.4 1397.22  3500.9 1393.54  3577.8 1383.23  3622.8 1380.99  3636.3  1383.3
  3676.9    1381  3742.7 1381.13  4066.9 1383.38  4334.8 1381.77  4793.4 1384.75
  4936.3 1388.81  4960.2  1385.6  4966.1 1379.57  4976.9 1374.92  4980.1  1371.8
  4980.6  1371.3  4998.8  1371.8  5001.2 1377.09  5021.8 1383.88  5057.9 1383.88
  5070.8 1386.18  5099.1 1397.17  5104.3 1403.44  5145.5 1416.74  5204.8 1425.65
#Mann= 9 ,-1 , 0
  3048.6     .12       0  3050.3     .07       0  3233.3     .12       0
  3286.2     .07       0  3742.7    .035       0  4334.8    .045       0
  4793.4    .035       0  4980.1     .05       0  4998.8     .12       0
Bank Sta=4980.1,4998.8
XS Rating Curve= 0 ,0
Exp/Cntr=0.3,0.1

Type RM Length L Ch R = 1 ,78645   ,765,765,765
BEGIN DESCRIPTION:
CURRY CREEK 123.0
END DESCRIPTION:
XS GIS Cut Line= 3
      2094022.31     13904973.05        2092925.       13902925.
      2092128.93     13902565.91
#Sta/Elev= 30
  2670.6 1418.42  2767.8 1414.58  2958.6  1408.2  3051.1 1405.25    3332 1394.28
  3353.9 1389.28  3419.7 1398.34  3451.2 1390.37    3540 1388.87  3567.6 1383.16
    3576 1389.67  3611.4 1384.99    3789 1381.45    3961 1379.18  4073.9 1378.59
  4463.8 1379.03  4488.9 1379.08  4878.5  1383.8  4942.1 1386.15    4986 1379.49
  4993.6 1370.19  4994.1 1369.69  5012.3 1370.19  5048.9 1380.55  5113.4 1384.54
  5222.1 1386.09  5249.8 1390.55  5393.7 1410.49  5516.1 1427.31  5867.4 1446.48
#Mann= 15 ,-1 , 0
  2670.6     .12       0  2767.8     .07       0  2958.6    .035       0
  3051.1     .07       0    3789    .035       0    3961     .07       0
  4073.9    .035       0  4463.8     .05       0  4488.9    .045       0
  4878.5    .035       0  4993.6    .035       0  5012.3    .035       0
  5113.4     .07       0  5249.8    .035       0  5393.7     .07       0
Bank Sta=4993.6,5012.3
XS Rating Curve= 0 ,0
Exp/Cntr=0.3,0.1

Type RM Length L Ch R = 1 ,77880   ,829,829,829
BEGIN DESCRIPTION:
Curry Creek 122.1
END DESCRIPTION:
XS GIS Cut Line= 3
      2094204.29     13904989.47      2093466.82     13902431.04
      2092698.73     13901761.11
#Sta/Elev= 30
  2337.4  1423.4  2473.8 1418.39  2633.7 1413.97  2747.1  1410.6  3054.4 1403.94
  3263.5 1398.07  3573.4 1380.85  3760.3  1377.3  3883.2 1376.82  3993.3  1377.1
  4366.7  1378.3  4408.1 1377.74  4501.1 1377.54  4698.8 1378.34  4839.1 1379.56
  4943.8 1383.17  4955.9 1371.67  4985.8 1366.84  4986.3 1366.34  5004.8 1366.84
  5033.8 1368.33  5062.3 1383.21  5293.7 1379.16    5367 1383.88  5508.5 1447.27
  5603.9 1437.63  5657.5 1431.09  5757.4 1448.61  5884.4 1456.23  6019.2 1452.05
#Mann= 20 ,-1 , 0
  2337.4     .12       0  2473.8     .07       0  2633.7     .12       0
  2747.1     .12       0  3054.4     .07       0  3263.5     .12       0
  3573.4     .07       0  3760.3    .035       0  3883.2     .07       0
  3993.3     .05       0  4366.7    .045       0  4408.1     .05       0
  4501.1    .045       0  4698.8    .045       0  4839.1    .035       0
  4985.8    .035       0  5004.8    .035       0  5293.7     .07       0
  5603.9    .035       0  5757.4     .07       0
Bank Sta=4985.8,5004.8
XS Rating Curve= 0 ,0
Exp/Cntr=0.3,0.1

Type RM Length L Ch R = 1 ,77051   ,659,659,659
BEGIN DESCRIPTION:
Curry Creek 122.0
END DESCRIPTION:
XS GIS Cut Line= 2
      2094401.78     13905026.74      2093978.71     13901299.98
#Sta/Elev= 30
  1827.4 1426.77    1915 1424.48  2188.3 1415.55  2352.3 1410.22  2451.7 1407.85
  2541.8 1405.77  3088.3 1398.64    3316  1381.7  3345.7 1380.56  3445.1 1379.18
  3544.4 1379.47  3801.6 1374.61  4056.8 1376.45  4339.5 1374.88  4720.2 1376.52
  4928.9 1377.86  4950.1 1373.58  4969.8 1361.92  4970.3 1361.42  4988.8 1361.92
  4999.4 1376.76  5059.6 1378.98  5124.3 1390.22  5190.6 1416.25  5208.9 1428.24
  5213.9 1426.37  5291.2 1466.71  5332.6 1472.31  5531.3 1474.04  5578.1 1473.05
#Mann= 19 ,-1 , 0
  1827.4     .07       0    1915     .12       0  2188.3     .07       0
  2352.3     .12       0  2451.7     .07       0  2541.8     .12       0
    3316    .035       0  3345.7     .07       0  3445.1    .035       0
  3544.4     .12       0  3801.6    .045       0  4056.8     .05       0
  4339.5    .045       0  4720.2    .035       0  4969.8    .035       0
  4988.8    .035       0  5059.6     .12       0  5332.6     .07       0
  5531.3    .035       0
Bank Sta=4969.8,4988.8
XS Rating Curve= 0 ,0
Exp/Cntr=0.3,0.1

Type RM Length L Ch R = 1 ,76392   ,790,790,790
BEGIN DESCRIPTION:
CURRY CREEK 121.0
END DESCRIPTION:
XS GIS Cut Line= 3
      2094773.31      13904513.4        2094625.       13902025.
      2094574.99     13901824.97
#Sta/Elev= 30
  2501.8 1414.58  2611.5 1410.08  2792.9 1403.82  3031.1 1396.23  3228.1 1386.16
  3386.2 1388.54  3402.9 1388.26  3441.9 1388.36  3582.7  1380.7  3742.4 1373.43
  3878.8 1371.26  3966.3 1371.14  4032.9 1372.13  4069.1 1368.64  4133.1 1373.08
    4175 1371.99    4664 1370.33  4944.5  1377.2  4964.6 1375.12  4974.6 1370.68
  4982.6 1359.84  4983.1 1359.34  5001.6 1359.84  5025.5 1361.44  5035.8 1370.88
  5046.2 1375.32    5059 1376.16  5065.9 1380.08  5095.1 1400.75  5200.8 1418.56
#Mann= 12 ,-1 , 0
  2501.8    .035       0  2611.5     .07       0  2792.9     .12       0
  3386.2     .07       0  3402.9     .12       0  3582.7     .07       0
  3878.8    .035       0  3966.3     .07       0    4175     .05       0
  4982.6     .05       0  5001.6     .05       0  5065.9     .12       0
Bank Sta=4982.6,5001.6
XS Rating Curve= 0 ,0
Exp/Cntr=0.3,0.1

Type RM Length L Ch R = 1 ,75602   ,561,561,561
BEGIN DESCRIPTION:
CURRY CREEK 120.0
END DESCRIPTION:
XS GIS Cut Line= 3
      2095034.33     13904296.13      2095231.05     13901626.67
      2094875.02     13901175.02
#Sta/Elev= 30
  2323.3 1408.28  2388.1 1406.32  2684.5 1397.77  2907.1 1390.54  2967.9 1388.39
  3026.3 1383.26  3331.8 1375.13  3563.7  1368.5  3792.7 1366.95  3915.4 1366.35
    4092 1366.53  4103.8 1366.49  4287.4 1366.66  4441.5 1367.56  4921.5 1373.04
  4931.5 1372.44  4951.5 1363.99  4962.1 1352.83  4962.6 1352.33  4981.1 1352.83
  4986.2 1352.97  4998.3 1371.78  5005.1 1373.24  5147.8 1367.99  5236.5 1369.76
  5269.5 1371.93  5346.6  1393.6  5435.5 1407.35  5468.5    1414  5575.1 1423.69
#Mann= 17 ,-1 , 0
  2323.3     .07       0  2388.1     .12       0  2684.5     .07       0
  2907.1     .12       0  2967.9    .035       0  3331.8     .07       0
  3563.7    .035       0  3792.7     .07       0  3915.4     .05       0
    4092     .07       0  4103.8     .05       0  4287.4     .07       0
  4441.5     .05       0  4962.1     .05       0  4981.1     .05       0
  5236.5     .07       0  5435.5     .12       0
Bank Sta=4962.1,4981.1
XS Rating Curve= 0 ,0
Exp/Cntr=0.3,0.1

Type RM Length L Ch R = 1 ,75041   ,822,822,822
BEGIN DESCRIPTION:
CURRY CREEK 119.0
END DESCRIPTION:
XS GIS Cut Line= 4
      2095495.35     13903538.75      2095721.62     13901766.82
        2095725.       13901525.      2095174.99     13901074.99
#Sta/Elev= 30
  2972.2 1394.13  3056.1 1390.55  3085.7 1390.29  3254.3 1384.02  3720.2 1369.65
  3792.6 1364.94    3798  1367.6    3803 1365.94  3812.7 1367.87  3878.6 1366.18
  4084.9 1365.72  4342.7 1365.58    4720 1364.89  4952.9  1369.5  4970.4 1366.68
  4997.9 1355.82  5003.6 1355.82  5004.5 1349.38    5005 1348.88  5023.5 1349.38
  5036.2 1358.82  5057.1 1368.82  5157.8 1366.77  5302.3 1365.65  5476.5 1365.94
  5518.6 1376.07    5576 1394.31  5625.6 1401.86  5654.9 1403.23    5711 1408.06
#Mann= 15 ,-1 , 0
  2972.2    .035       0  3056.1     .07       0  3085.7    .035       0
  3254.3     .12       0  3720.2     .07       0  3878.6     .05       0
  4084.9     .07       0  4342.7     .05       0  4952.9     .07       0
  5004.5     .05       0  5023.5     .07       0  5157.8     .07       0
  5302.3     .05       0  5476.5     .12       0  5654.9     .07       0
Bank Sta=5004.5,5023.5
XS Rating Curve= 0 ,0
Exp/Cntr=0.3,0.1

Type RM Length L Ch R = 1 ,74219   ,259,259,259
BEGIN DESCRIPTION:
CURRY CREEK 118.0
END DESCRIPTION:
XS GIS Cut Line= 3
      2097043.68     13902181.05        2096325.       13901425.
      2095259.76     13901013.43
#Sta/Elev= 30
  3956.5 1386.18  3967.5 1385.45  4094.2 1371.73  4170.1 1369.52  4244.7 1366.12
  4309.9 1364.19  4383.2  1362.2  4449.7 1361.39  4521.8 1361.59  4660.4 1361.67
  4825.5 1361.24  4957.3 1362.96  4971.5 1347.96  4980.5 1346.49    4981 1345.99
  5004.5 1346.49  5014.6 1347.37  5044.6 1363.06  5057.2  1365.2  5129.1 1363.12
  5266.1  1365.2  5401.8 1366.99  5474.9 1365.16  5617.9 1365.93  5803.7 1362.69
  5921.6 1364.06  5968.3 1367.33  6050.2 1392.68  6121.6 1403.08  6141.6 1403.34
#Mann= 17 ,-1 , 0
  3956.5     .12       0  3967.5    .035       0  4170.1     .12       0
  4244.7    .035       0  4309.9     .07       0  4383.2    .035       0
  4449.7     .07       0  4521.8     .12       0  4660.4    .035       0
  4825.5     .07       0  4980.5     .05       0  5004.5     .07       0
  5057.2     .05       0  5266.1     .07       0  5474.9    .045       0
  5617.9     .05       0  5968.3     .12       0
Bank Sta=4980.5,5004.5
XS Rating Curve= 0 ,0
Exp/Cntr=0.3,0.1

Type RM Length L Ch R = 1 ,73960   ,493,493,493
BEGIN DESCRIPTION:
CURRY CREEK 117.0
END DESCRIPTION:
XS GIS Cut Line= 3
        2096925.       13901825.      2096527.18     13901471.68
      2095775.02     13899875.04
#Sta/Elev= 30
  4474.2 1379.61  4572.2 1372.88  4619.3 1371.01  4700.5 1366.58  4772.7 1361.52
  4934.6 1361.97  4957.2 1357.17    4963  1357.5  4983.9 1346.04  4991.4 1348.11
  5001.6 1344.58  5002.1 1344.08  5025.6 1344.58  5026.6 1346.78  5035.8 1348.96
  5043.9  1358.3  5089.5 1361.59  5279.7 1361.06  5510.1  1360.1  5759.1 1357.63
  6425.8 1353.56  6523.7 1353.78  6546.5 1357.31    6560 1354.38  6574.8 1353.31
  6620.4 1368.71  6643.2 1378.65  6688.7 1407.13  6747.3 1427.53  6771.2 1431.09
#Mann= 15 ,-1 , 0
  4474.2     .07       0  4572.2     .12       0  4619.3     .07       0
  4700.5     .12       0  4772.7     .07       0  4957.2    .035       0
  5001.6    .035       0  5025.6    .035       0  5026.6     .07       0
  5279.7    .045       0  5510.1     .07       0  5759.1    .045       0
  6425.8    .035       0    6560     .12       0  6747.3     .07       0
Bank Sta=5001.6,5025.6
XS Rating Curve= 0 ,0
Exp/Cntr=0.3,0.1

Type RM Length L Ch R = 1 ,73467   ,537,537,537
BEGIN DESCRIPTION:
CURRY CREEK 116.0
END DESCRIPTION:
XS GIS Cut Line= 3
      2097141.77     13901509.88        2096775.       13901125.
      2095925.01     13899525.02
#Sta/Elev= 30
  4462.4 1373.89  4739.4 1365.97  4781.7 1361.78  4831.3 1356.84  4951.8 1358.81
  4960.8 1342.48  4961.3 1341.98  4984.9 1342.48  5002.2 1345.41  5007.9 1356.92
  5042.6 1359.35  5417.2 1356.53  5429.7 1356.21  6170.2 1351.59  6296.3 1352.75
  6309.1 1356.01  6331.1 1351.03  6341.6 1354.45  6348.1 1359.24  6391.3 1372.68
  6451.6 1401.65  6457.3 1406.38  6488.8  1413.1  6495.6 1417.25  6523.2 1425.31
  6576.2 1431.78  6627.5 1440.39  6678.5 1444.38  6726.1 1454.14  6805.8 1461.18
#Mann= 11 ,-1 , 0
  4462.4     .12       0  4781.7    .035       0  4960.8    .035       0
  4984.9    .035       0  5042.6    .045       0  5417.2     .07       0
  5429.7    .045       0  6170.2     .07       0  6348.1     .12       0
  6576.2     .07       0  6678.5    .035       0
Bank Sta=4960.8,4984.9
XS Rating Curve= 0 ,0
Exp/Cntr=0.3,0.1

Type RM Length L Ch R = 1 ,72930   ,612,612,612
BEGIN DESCRIPTION:
CURRY CREEK 115.0
END DESCRIPTION:
XS GIS Cut Line= 3
      2097224.98     13901024.97        2097025.       13900675.
        2096025.       13899375.
#Sta/Elev= 30
  4596.7 1369.13  4794.9 1364.97  4890.2 1356.82  4948.7 1356.13  4954.4 1347.76
  4964.5 1344.28  4964.7 1338.74  4965.2 1338.24  4988.8 1338.74  5002.9 1341.39
  5013.3 1352.75  5027.8 1357.52  5066.5 1355.89    5382 1352.62  5955.8 1349.41
  5997.4 1354.24  6020.1 1349.78  6026.4 1351.16  6040.9 1363.51  6052.4 1367.22
  6105.3 1379.23  6111.6 1376.71  6169.6  1394.7  6214.1 1397.19  6254.8 1398.88
  6308.3 1407.29  6461.5 1441.22  6482.4 1445.51    6504  1452.3  6639.9 1471.29
#Mann= 12 ,-1 , 0
  4596.7     .12       0  4794.9     .07       0  4890.2    .035       0
  4964.7    .035       0  4988.8    .035       0  5066.5    .045       0
    5382     .07       0  6052.4     .12       0  6214.1     .07       0
  6308.3    .035       0  6461.5     .07       0  6482.4    .035       0
Bank Sta=4964.7,4988.8
XS Rating Curve= 0 ,0
Exp/Cntr=0.3,0.1

Type RM Length L Ch R = 1 ,72318   ,434,434,434
BEGIN DESCRIPTION:
CURRY CREEK 114.0
END DESCRIPTION:
XS GIS Cut Line= 3
        2097725.     13900724.99      2097197.32     13900159.18
      2096374.97     13899424.97
#Sta/Elev= 30
  4221.7  1361.9  4306.5 1359.34  4342.1 1355.16  4433.2 1351.62  4490.6 1350.56
    4519 1347.97  4571.9 1351.42  4740.3 1350.98  4823.6 1351.05  4879.5 1350.16
  4936.2 1352.03  4943.5 1347.04  4950.4 1336.83  4957.7 1338.39  4983.3 1335.19
  4983.8 1334.69  5007.4 1335.19  5013.9  1339.4  5021.4 1352.61  5028.1 1353.34
  5092.3 1350.24  5299.5    1349  5639.1 1348.23  5672.7 1352.05  5686.9 1347.59
  5694.4 1347.37  5757.9 1373.11  5901.7 1411.89  5963.6 1423.43  6097.8 1436.69
#Mann= 10 ,-1 , 0
  4221.7     .12       0  4433.2     .07       0  4571.9    .035       0
  4740.3     .07       0  4823.6    .035       0  4983.3    .045       0
  5007.4    .035       0  5299.5     .07       0  5639.1     .12       0
  5901.7     .07       0
Bank Sta=4983.3,5007.4
XS Rating Curve= 0 ,0
Exp/Cntr=0.3,0.1

Type RM Length L Ch R = 1 ,71884   ,597,597,597
BEGIN DESCRIPTION:
CURRY CREEK 113.0
END DESCRIPTION:
XS GIS Cut Line= 3
        2097725.       13900675.      2097471.62      13899881.4
      2096774.99     13899074.99
#Sta/Elev= 30
  4157.9 1360.32  4317.3 1349.47  4367.1 1349.97  4420.3 1346.75  4474.2 1349.84
  4527.2  1347.8    4802 1348.36  4962.2 1350.61  4967.4 1348.37  4976.7 1339.31
  4986.4 1334.82  5001.9  1333.8  5002.4  1333.3    5026  1333.8  5028.2 1340.05
  5035.9 1349.88  5139.5  1347.6  5396.8 1344.23  5425.3 1345.44  5439.6 1348.68
  5453.8 1344.79  5527.2  1355.9  5730.3 1371.08  5794.2 1379.05    5821 1382.77
  5893.7 1394.43  5943.1 1398.28  5978.2 1406.55    6021    1411  6056.6 1418.26
#Mann= 10 ,-1 , 0
  4157.9     .12       0  4317.3     .07       0  4527.2    .035       0
    4802     .07       0  5001.9     .05       0    5026     .07       0
  5139.5    .045       0  5527.2     .12       0  5794.2     .07       0
    5821    .035       0
Bank Sta=5001.9,5026
XS Rating Curve= 0 ,0
Exp/Cntr=0.3,0.1

Type RM Length L Ch R = 1 ,71287   ,863,863,863
BEGIN DESCRIPTION:
CURRY CREEK 112.0
END DESCRIPTION:
XS GIS Cut Line= 3
        2097825.     13900625.02        2097975.       13899825.
      2097175.02     13899025.02
#Sta/Elev= 30
  4186.5 1357.42  4205.1 1356.85  4326.2 1352.11    4624 1345.07  4695.9 1344.97
  4897.8 1347.41  4908.9 1348.04  4916.5 1344.89  4921.6 1348.27  4929.2 1339.71
  4939.4 1335.05  4962.1  1330.5  4962.6    1330  4986.2  1330.5  4990.3 1336.49
  4997.9 1341.77  5029.4 1347.36  5062.4 1345.98  5173.1 1344.85  5403.2 1343.58
  5471.9 1343.37  5513.1 1343.01  5580.3 1343.19  5594.4 1338.83  5608.6 1344.37
  5707.6    1347  5867.6 1357.12    5948  1364.3    6054 1381.09  6131.8 1391.94
#Mann= 15 ,-1 , 0
  4186.5     .07       0  4205.1     .12       0  4326.2     .07       0
  4695.9    .035       0  4897.8     .07       0  4962.1     .05       0
  4986.2     .07       0  5029.4    .035       0  5062.4     .07       0
  5173.1    .045       0  5403.2    .035       0  5471.9    .045       0
  5513.1    .035       0  5867.6     .07       0    6054     .12       0
Bank Sta=4962.1,4986.2
XS Rating Curve= 0 ,0
Exp/Cntr=0.3,0.1

Type RM Length L Ch R = 1 ,70424   ,799,799,799
BEGIN DESCRIPTION:
Curry Creek 111.1
END DESCRIPTION:
XS GIS Cut Line= 3
      2099227.96      13900800.1      2098229.39     13899106.73
      2097696.03     13898716.06
#Sta/Elev= 30
  3045.9 1373.75    3241 1365.85  3293.8 1365.53  3401.1  1356.6  3570.9 1348.77
  4146.6 1341.17  4162.3 1337.28  4189.5 1335.78  4328.8 1342.98  4372.1 1341.63
  4723.5 1342.46  4892.2 1340.93  4956.5 1342.32  4966.4 1340.71  4966.5 1327.51
    4967 1327.01  4991.4 1327.51  5002.2  1327.9  5011.8 1331.68  5017.5 1331.68
  5023.3 1340.59  5029.6 1341.81  5119.1 1340.56  5265.7 1340.25  5311.6 1343.05
    5339 1348.55  5401.6 1368.28  5481.1 1387.12  5552.1  1392.5  5672.9 1392.07
#Mann= 7 ,-1 , 0
  3045.9    .035       0    3241     .07       0  4372.1    .035       0
  4966.5     .05       0  4991.4    .035       0  5119.1     .07       0
  5311.6     .12       0
Bank Sta=4966.5,4991.4
XS Rating Curve= 0 ,0
Exp/Cntr=0.3,0.1

Type RM Length L Ch R = 1 ,69625   ,849,849,849
BEGIN DESCRIPTION:
Curry Creek 111.0
END DESCRIPTION:
XS GIS Cut Line= 3
      2099394.63     13900745.34      2098566.56     13898424.77
      2098233.67     13897953.47
#Sta/Elev= 30
  2542.6 1370.77  2824.3 1363.85  2935.8 1357.14  2978.3 1352.25  3096.2 1346.91
  3381.8 1341.22  3716.5 1338.16    3764 1333.12  3871.3 1336.01  4490.9 1338.39
  4687.7 1335.09    4792 1336.66  4962.5 1337.69  4967.8 1337.18  4974.4 1328.98
    4985  1324.6  5002.6 1321.43  5003.1 1320.93  5027.5 1321.43  5029.9  1328.4
  5042.9 1342.66  5064.7  1350.7  5086.5 1356.53  5107.4 1367.53  5178.8 1386.54
  5228.4 1387.96  5279.8 1387.53  5379.2 1380.77  5462.8 1374.77  5583.5  1371.4
#Mann= 9 ,-1 , 0
  2542.6     .07       0  3871.3    .035       0    4792     .07       0
  5002.6     .05       0  5027.5     .07       0  5064.7     .12       0
  5228.4     .07       0  5379.2     .12       0  5462.8     .07       0
Bank Sta=5002.6,5027.5
XS Rating Curve= 0 ,0
Exp/Cntr=0.3,0.1

Type RM Length L Ch R = 1 ,68776   ,793,793,793
BEGIN DESCRIPTION:
Curry Creek 110.0
END DESCRIPTION:
XS GIS Cut Line= 4
      2099454.58     13900632.28      2099308.94     13898750.36
      2099211.25     13897974.27      2098577.05     13897278.62
#Sta/Elev= 30
  2330.9    1368  2569.4 1363.35  2704.3 1350.75  2799.6 1345.06  3672.2 1333.75
  3712.3 1330.76  4044.9 1332.39    4114 1331.83  4212.9 1331.08  4312.4 1329.84
  4909.5 1332.15  4949.5 1332.88  4959.6 1325.23  4977.3 1319.48  4977.8 1318.98
  5002.3 1319.48  5012.2 1325.08  5026.1 1333.61  5032.8 1333.77  5040.3 1342.11
  5061.2 1350.06    5068 1347.87  5087.6 1351.74  5224.1 1351.69  5358.5 1342.53
  5429.4 1343.24  5620.6 1356.09  5634.8 1354.36  5832.8 1373.89    5942 1381.05
#Mann= 12 ,-1 , 0
  2330.9     .07       0  2569.4     .12       0  2704.3     .07       0
  4044.9     .12       0    4114    .035       0  4212.9     .07       0
  4312.4    .035       0  4909.5     .07       0  4977.3     .05       0
  5002.3     .07       0  5012.2     .12       0  5087.6     .07       0
Bank Sta=4977.3,5002.3
XS Rating Curve= 0 ,0
Exp/Cntr=0.3,0.1

Type RM Length L Ch R = 1 ,67983   ,644,644,644
BEGIN DESCRIPTION:
Curry Creek 109.0
END DESCRIPTION:
XS GIS Cut Line= 3
      2100137.19     13900072.37        2099925.       13898125.
      2099815.55     13897098.32
#Sta/Elev= 30
  3041.1 1363.34  3249.8 1350.61  3327.5 1348.13  3450.6 1346.12  3662.3 1334.68
  3796.4 1330.58  3847.7  1330.3  3984.3 1328.29    4097 1327.15  4165.1 1325.34
    4258 1327.96  4386.2 1328.06  4528.7 1326.12  4857.8 1324.45  4938.9  1327.6
  4959.8 1328.29    4985 1315.64  4985.5 1315.14    5010 1315.64  5046.2 1328.99
  5138.3 1325.71  5281.6 1325.17  5333.5 1330.11  5376.7  1340.4  5452.6  1349.9
  5512.9  1351.4  5579.6  1358.5    5714 1376.64  5925.2 1393.14  6032.5 1395.42
#Mann= 18 ,-1 , 0
  3041.1     .07       0  3249.8    .035       0  3327.5     .07       0
  3450.6     .12       0  3662.3     .07       0  3796.4    .035       0
  3847.7     .07       0  3984.3    .035       0    4097     .07       0
    4258    .035       0  4386.2     .07       0  4528.7    .035       0
  4938.9     .07       0    4985     .05       0    5010     .07       0
  5138.3    .035       0  5376.7     .12       0  5579.6     .07       0
Bank Sta=4985,5010
XS Rating Curve= 0 ,0
Exp/Cntr=0.3,0.1

Type RM Length L Ch R = 1 ,67339   ,692,692,692
BEGIN DESCRIPTION:
Curry Creek 108.0
END DESCRIPTION:
XS GIS Cut Line= 3
      2101011.48     13899961.75      2100481.41     13897870.44
      2100305.05     13897499.58
#Sta/Elev= 30
  2840.9 1369.09  2867.7 1368.21  3002.6 1361.85  3023.2 1358.44  3105.8 1353.87
  3363.7 1346.03  3425.6 1340.22  3500.5 1337.33  3577.3 1330.68  3582.5 1332.12
  3659.3 1328.75  3879.2 1324.99  4432.8 1323.49  4790.4 1322.32  4795.5 1322.25
  4878.5    1322  4924.6 1324.21  4942.1 1322.86  4970.8 1314.86  4971.3 1314.36
  4995.8 1314.86  5037.6 1323.26  5080.9 1323.54    5104 1321.44  5158.2  1322.4
  5181.5 1321.28  5215.7 1327.54  5301.1 1332.87  5358.7  1340.3    5409 1344.35
#Mann= 10 ,-1 , 0
  2840.9     .12       0  2867.7     .07       0  3879.2    .035       0
  4432.8     .07       0  4790.4    .035       0  4795.5     .07       0
  4970.8     .05       0  4995.8     .07       0  5080.9    .035       0
  5158.2     .12       0
Bank Sta=4970.8,4995.8
XS Rating Curve= 0 ,0
Exp/Cntr=0.3,0.1

Type RM Length L Ch R = 1 ,66647   ,902,902,902
BEGIN DESCRIPTION:
Curry Creek 107.0
END DESCRIPTION:
XS GIS Cut Line= 3
      2101650.03     13898300.04        2100975.       13897425.
      2100219.57      13896796.4
#Sta/Elev= 30
  3889.5 1340.01  3970.3 1339.34  3982.7 1339.25  4103.3 1338.79  4248.6 1333.96
  4340.6 1331.97  4444.4 1328.21    4539 1325.65  4590.3 1314.23  4590.8 1313.73
  4615.9 1314.23  4629.2 1316.05  4733.8 1318.55  4758.6 1318.82  4913.7 1318.12
  4944.1 1317.22  4981.1 1316.69  4988.3 1316.04  5054.5 1320.85  5171.4 1319.93
  5242.7 1318.58  5335.1    1322  5413.2 1333.91  5470.5 1348.51  5555.1 1354.37
  5657.4 1366.08  5711.3 1375.81  5772.3 1380.56  5924.8 1394.99  5977.4 1396.16
#Mann= 19 ,-1 , 0
  3889.5     .07       0  3970.3     .12       0  3982.7     .07       0
  4248.6     .12       0  4340.6     .07       0  4444.4     .12       0
  4590.3     .05       0  4615.9     .12       0  4629.2     .07       0
  4733.8     .12       0  4758.6     .12       0  4913.7    .035       0
  4944.1    .035       0  4981.1     .07       0  4988.3     .07       0
  5054.5    .035       0  5171.4     .07       0  5657.4    .035       0
  5772.3     .07       0
Bank Sta=4944.1,4981.1
XS Rating Curve= 0 ,0
Exp/Cntr=0.3,0.1

Type RM Length L Ch R = 1 ,65745   ,635,635,635
BEGIN DESCRIPTION:
CURRY CREEK 106.0
END DESCRIPTION:
XS GIS Cut Line= 3
      2101724.98     13897024.99        2101375.       13896825.
      2101025.01     13896325.02
#Sta/Elev= 30
  4596.2  1325.6  4703.6 1321.98  4743.7 1318.97  4808.5 1320.26  4824.4 1315.17
  4831.6 1315.03    4838 1312.21  4861.1  1310.8    4898 1315.18  4910.8 1317.22
  4953.9  1311.8    4964 1305.91  4976.3 1302.81  4978.2 1299.97  4978.7 1299.47
  5004.6 1299.97  5006.7    1306  5012.8 1310.18  5027.6 1313.08  5093.6 1311.67
  5179.7 1312.92  5386.1 1313.99  5456.4 1314.96  5487.6 1319.37  5524.2 1336.59
  5530.7 1342.04  5545.5 1346.13  5551.6 1351.35  5560.4 1353.79  5609.6 1356.77
#Mann= 10 ,-1 , 0
  4596.2     .12       0  4703.6     .07       0  4831.6    .035       0
    4898     .07       0  4978.2     .05       0  5004.6     .07       0
  5093.6    .035       0  5179.7     .07       0  5386.1    .035       0
  5456.4     .12       0
Bank Sta=4978.2,5004.6
XS Rating Curve= 0 ,0
Exp/Cntr=0.3,0.1

Type RM Length L Ch R = 1 ,65110   ,414,414,414
BEGIN DESCRIPTION:
Curry Creek 105.0
END DESCRIPTION:
XS GIS Cut Line= 3
      2102014.49     13896922.58      2101688.45      13896319.8
      2101480.06     13896044.73
#Sta/Elev= 30
  4272.6 1326.16  4338.1 1324.66  4394.9 1317.81  4444.4 1315.36  4485.9 1313.81
    4520 1308.06  4558.9 1311.69  4672.7 1311.43  4748.7 1309.62  4786.4 1306.83
    4803 1305.76  4834.8 1308.33  4918.1 1308.81  4934.3 1307.65  4956.2 1299.91
  4972.3 1298.65  4972.8 1298.15  4998.9 1298.65  5000.2 1303.24  5016.2 1305.99
  5070.9 1306.97  5091.7 1313.13  5106.3 1320.45  5114.5 1330.56  5120.8 1341.01
  5127.1 1342.04  5135.4 1357.45  5146.4 1358.61  5272.7 1364.38    5303 1365.24
#Mann= 11 ,-1 , 0
  4272.6     .12       0  4444.4     .07       0  4558.9    .035       0
  4672.7     .12       0  4786.4     .07       0  4834.8     .12       0
  4972.3     .05       0  4998.9     .12       0  5016.2     .07       0
  5146.4     .12       0  5272.7     .07       0
Bank Sta=4972.3,4998.9
XS Rating Curve= 0 ,0
Exp/Cntr=0.3,0.1

Type RM Length L Ch R = 1 ,64696   ,575,575,575
BEGIN DESCRIPTION:
CURRY CREEK 104.0
END DESCRIPTION:
XS GIS Cut Line= 3
      2102125.01     13896875.04        2102025.       13896225.
        2101825.       13895875.
#Sta/Elev= 30
  4346.6 1325.77  4397.2 1323.36  4427.6 1318.66  4488.3 1314.16  4507.3 1308.33
  4528.4 1308.24  4569.2 1311.42  4802.6 1308.26  4882.9 1306.05  4933.5    1307
  4963.8 1300.87  4970.8 1295.39  4971.3 1294.89  4997.4 1295.39  5001.8 1302.37
  5004.6 1302.37  5008.4 1303.13    5018 1305.94  5033.8 1304.21  5055.4 1305.84
    5077 1311.52  5092.8 1324.87  5098.6 1324.91  5114.4  1332.9    5136  1337.8
  5179.2 1353.91  5232.5 1359.57  5283.7 1360.92  5334.7 1367.69  5407.4 1370.92
#Mann= 8 ,-1 , 0
  4346.6     .12       0  4528.4     .07       0  4802.6     .12       0
  4970.8     .05       0  4997.4     .12       0  5004.6     .07       0
  5008.4     .12       0  5283.7     .07       0
Bank Sta=4970.8,4997.4
XS Rating Curve= 0 ,0
Exp/Cntr=0.3,0.1

Type RM Length L Ch R = 1 ,64121   ,711,711,711
BEGIN DESCRIPTION:
CURRY CREEK 103.0
END DESCRIPTION:
XS GIS Cut Line= 3
      2102375.01     13896824.96        2102525.       13896025.
      2102325.01     13895675.01
#Sta/Elev= 30
  4186.1 1324.81  4243.4 1318.52  4314.9  1312.1  4321.7 1311.85  4328.5 1306.15
    4359 1313.28  4369.2 1313.36  4389.5 1312.72  4399.7 1309.44  4420.1 1307.34
  4525.7 1307.12  4648.1 1306.49  4684.6 1298.69  4715.1 1299.06  4735.5 1302.54
  4829.3 1305.26  4959.3 1304.27  4968.6 1301.81  4973.7 1303.58  4989.8 1297.94
  4994.6 1293.13  4995.1 1292.63  5021.2 1293.13    5027 1293.93  5045.3 1300.63
  5080.6 1300.29  5147.6 1329.95  5190.8 1340.11  5299.5 1350.56  5403.1 1354.21
#Mann= 8 ,-1 , 0
  4186.1     .12       0  4243.4     .07       0  4314.9     .12       0
  4525.7    .035       0  4829.3     .07       0  4994.6     .05       0
  5021.2     .07       0    5027     .12       0
Bank Sta=4994.6,5021.2
XS Rating Curve= 0 ,0
Exp/Cntr=0.3,0.1

Type RM Length L Ch R = 1 ,63410   ,293,293,293
BEGIN DESCRIPTION:
Curry Creek 102.0
END DESCRIPTION:
XS GIS Cut Line= 3
      2102508.71     13896894.41      2103185.71     13895876.72
      2102784.48     13895265.43
#Sta/Elev= 30
  3777.7 1323.56  3795.6 1322.15  3961.9 1313.67  4018.2 1306.23  4127.2  1315.1
  4163.3 1314.75  4172.3 1311.61  4178.3 1314.14  4193.3 1308.12  4200.1 1309.43
  4244.4 1305.96  4663.5 1300.03  4828.7 1298.54  4899.7 1297.33  4995.9 1290.07
  4996.4 1289.57  5022.6 1290.07  5024.3  1296.4  5030.3 1297.77  5066.5 1299.95
  5267.7 1302.82  5319.6 1308.09  5325.6 1312.12  5334.7 1311.97  5340.7 1317.88
  5370.9    1320  5397.9 1329.73  5453.3 1333.79  5707.8 1346.27  5731.2 1348.54
#Mann= 11 ,-1 , 0
  3777.7     .12       0  3795.6     .07       0  4018.2     .12       0
  4200.1    .035       0  4663.5     .07       0  4828.7     .12       0
  4995.9     .05       0  5022.6     .12       0  5267.7     .12       0
  5453.3     .07       0  5707.8    .035       0
Bank Sta=4995.9,5022.6
XS Rating Curve= 0 ,0
Exp/Cntr=0.3,0.1

Type RM Length L Ch R = 1 ,63117   ,383,383,383
BEGIN DESCRIPTION:
Curry Creek 101.5
END DESCRIPTION:
XS GIS Cut Line= 3
      2104284.39      13896097.6      2103405.76     13895694.23
      2102852.82     13895053.81
#Sta/Elev= 30
  4033.2 1333.57  4058.6 1333.34  4208.7 1330.44  4315.6 1313.61  4392.7 1308.61
  4529.5 1304.92  4636.4 1302.03  4703.9 1299.89  4813.3  1288.5  4841.8 1292.81
  4879.8 1291.38  4897.4 1295.15  4931.2 1296.54  4962.3 1295.32  4967.8 1290.74
  4984.3 1286.73  4984.8 1286.23    5011 1286.73  5013.8 1294.13  5035.9 1297.02
  5213.1 1300.91    5233 1300.74  5312.2  1302.9  5326.4 1306.23  5368.9 1326.48
  5414.8 1330.57  5613.6 1337.97  5669.9 1341.07  5726.7 1345.12  5846.1 1353.67
#Mann= 18 ,-1 , 0
  4033.2     .07       0  4058.6     .12       0  4208.7     .07       0
  4315.6    .035       0  4392.7     .07       0  4529.5    .035       0
  4636.4     .07       0  4897.4    .035       0  4931.2     .07       0
  4984.3     .05       0    5011     .07       0  5035.9    .035       0
  5213.1     .07       0    5233     .12       0  5414.8     .07       0
  5613.6    .035       0  5669.9     .07       0  5726.7    .035       0
Bank Sta=4984.3,5011
XS Rating Curve= 0 ,0
Exp/Cntr=0.3,0.1

Type RM Length L Ch R = 1 ,62734   ,343,343,343
BEGIN DESCRIPTION:
Curry Creek 101.0
END DESCRIPTION:
XS GIS Cut Line= 2
      2104268.13     13895853.07      2103273.03     13895199.39
#Sta/Elev= 30
  4300.8 1329.29  4344.6 1328.39  4401.9 1320.12    4438 1317.43  4477.9 1310.39
  4546.5 1305.62  4699.4 1303.06  4735.3 1301.27  4799.6 1301.17    4870 1297.99
  4886.8 1297.28  4944.3 1297.58  4974.4 1289.58  4983.2 1283.85  4984.1 1283.35
  5019.7 1283.85  5022.6 1289.77  5040.5  1292.6  5041.7 1292.67  5094.9 1295.41
  5129.1 1294.42  5167.2 1295.55  5197.4 1293.84  5248.6 1297.98  5311.8 1299.59
  5340.1 1303.69  5393.3 1305.31  5441.4 1315.03  5465.1 1316.88  5491.4 1323.18
#Mann= 10 ,-1 , 0
  4300.8     .07       0  4477.9    .035       0    4870     .07       0
  4886.8    .035       0  4983.2    .035       0  5019.7    .035       0
  5040.5     .07       0  5041.7    .035       0  5129.1     .07       0
  5340.1     .12       0
Bank Sta=4983.2,5019.7
XS Rating Curve= 0 ,0
Exp/Cntr=0.3,0.1

Type RM Length L Ch R = 1 ,62391   ,540,540,540
BEGIN DESCRIPTION:
CURRY CREEK 100.0
END DESCRIPTION:
XS GIS Cut Line= 3
      2104474.97     13895474.99        2103825.       13895175.
        2103175.       13894825.
#Sta/Elev= 30
  4283.9 1327.16    4321 1326.07  4389.9 1319.36  4431.6 1310.18  4493.1 1300.83
    4768 1298.31  4903.7 1295.26  4933.7 1295.02  4939.6  1292.8  4944.3 1282.88
  4945.2 1282.38  4980.9 1282.88    4991 1285.92  5013.5 1283.32  5022.5 1285.53
  5035.5  1291.7  5056.7 1292.92  5075.9 1293.33  5139.3 1291.28  5215.6 1293.65
  5272.3 1299.24  5324.2 1300.13  5374.1 1303.35  5478.4 1311.92  5494.6 1315.64
  5538.4 1320.92  5554.7 1326.01  5620.4 1337.64  5702.3 1346.98    5738 1347.88
#Mann= 9 ,-1 , 0
  4283.9     .07       0  4431.6    .035       0  4903.7     .07       0
  4944.3     .05       0  4980.9     .07       0  5056.7    .035       0
  5075.9     .07       0  5324.2     .12       0  5374.1     .07       0
Bank Sta=4944.3,4980.9
XS Rating Curve= 0 ,0
Exp/Cntr=0.3,0.1

Type RM Length L Ch R = 1 ,61851   ,571,571,571
BEGIN DESCRIPTION:
CURRY CREEK 99.0
END DESCRIPTION:
XS GIS Cut Line= 3
      2104575.01     13895075.01        2104225.       13894825.
      2103425.03     13894325.02
#Sta/Elev= 30
  4569.9 1326.54    4592 1325.36  4606.8 1320.72  4644.2 1319.56  4685.7 1317.64
  4705.1    1314  4713.7 1310.63  4734.6 1307.61  4749.3 1301.76  4764.1 1298.61
  4838.9 1295.17  4950.9 1292.58  4971.8  1287.6  4989.4 1280.38  4990.3 1279.88
    5026 1280.38  5028.9 1286.47  5071.4 1285.46  5116.1 1289.19  5211.7 1291.83
  5247.7 1290.27  5268.1 1292.52  5318.4 1295.92  5635.1  1300.3  5710.5 1301.68
  5783.6 1311.39  5856.8 1332.67  5879.2 1336.88  5899.2 1340.87  5943.4 1344.66
#Mann= 10 ,-1 , 0
  4569.9     .07       0  4644.2     .12       0  4685.7     .07       0
  4838.9    .035       0  4989.4    .035       0    5026    .035       0
  5116.1     .12       0  5268.1    .035       0  5635.1     .07       0
  5879.2     .12       0
Bank Sta=4989.4,5026
XS Rating Curve= 0 ,0
Exp/Cntr=0.3,0.1

Type RM Length L Ch R = 1 ,61280   ,566,566,566
BEGIN DESCRIPTION:
CURRY CREEK 98.0
END DESCRIPTION:
XS GIS Cut Line= 3
      2104674.98     13894774.97        2104425.       13894325.
      2103724.98     13893924.99
#Sta/Elev= 30
  4485.4 1317.51  4522.1 1316.57  4542.6 1313.44  4602.1 1308.87  4714.2 1304.78
  4805.1 1296.84  4883.5 1293.18  4889.2 1291.71  4926.8 1290.76  4932.7 1286.53
    4943 1285.15  4954.4  1279.4  4986.4 1277.67  4989.8 1276.42  4990.6 1275.92
  5026.4 1276.42  5029.7 1282.96  5057.7 1286.08  5094.4 1285.58  5175.1 1293.07
  5206.7 1293.28  5255.7 1295.88  5590.1 1294.11  5622.1 1294.75  5637.2 1297.11
  5696.2 1315.52  5717.8 1325.11  5739.4    1330  5776.9 1334.43  5806.4 1335.67
#Mann= 7 ,-1 , 0
  4485.4     .07       0  4522.1     .12       0  4805.1     .07       0
  4926.8    .035       0  4989.8    .035       0  5026.4    .035       0
  5590.1     .12       0
Bank Sta=4989.8,5026.4
XS Rating Curve= 0 ,0
Exp/Cntr=0.3,0.1

Type RM Length L Ch R = 1 ,60714   ,365,365,365
BEGIN DESCRIPTION:
CURRY CREEK 97.0
END DESCRIPTION:
XS GIS Cut Line= 3
      2104974.98     13894624.96        2104575.       13893825.
      2103229.25     13893536.07
#Sta/Elev= 30
  4105.3 1317.58  4223.2 1307.66  4327.5    1303    4382  1297.5  4466.8 1294.92
  4767.7  1292.3  4798.5 1288.25  4963.4 1280.63  4991.6 1275.16  4992.5 1274.66
  5028.2 1275.16  5030.4 1282.87  5061.1 1281.57  5187.9 1289.55  5503.8 1290.11
  5591.5 1293.38  5633.8 1306.84  5674.7 1325.16  5690.3 1327.72    5799 1331.03
  5991.8  1331.5  6012.2 1329.05  6053.2 1312.84  6094.1 1307.71  6114.3 1310.84
  6124.8  1318.4  6163.7 1331.06  6189.4 1335.04  6218.4 1336.46  6376.1 1342.65
#Mann= 12 ,-1 , 0
  4105.3     .07       0  4223.2    .035       0  4327.5     .07       0
  4466.8    .035       0  4798.5     .07       0  4991.6     .05       0
  5028.2     .07       0  5187.9    .035       0  5503.8     .12       0
    5799     .07       0  6189.4     .12       0  6218.4     .07       0
Bank Sta=4991.6,5028.2
XS Rating Curve= 0 ,0
Exp/Cntr=0.3,0.1

Type RM Length L Ch R = 1 ,60349   ,748,748,748
BEGIN DESCRIPTION:
CURRY CREEK 96.0
END DESCRIPTION:
XS GIS Cut Line= 3
      2105174.98     13894424.96      2104858.78     13893624.46
      2103780.63     13892676.53
#Sta/Elev= 30
  4139.4 1316.27  4154.5 1315.59  4322.1 1290.75  4354.4 1289.21  4747.2 1290.31
  4795.2 1289.27  4827.5 1283.28  4956.5 1280.84  4971.1 1278.64  4979.9 1273.17
  4980.8 1272.67    5017 1273.17  5023.5 1277.49  5037.8 1278.81  5089.1  1279.8
  5139.7 1282.27  5158.3 1279.24  5164.9  1283.2  5271.4 1284.15  5344.6 1289.53
  5472.4 1291.63  5478.9 1291.89  5787.6 1308.08  5859.5 1315.22    6016 1319.14
  6143.1 1331.98    6275  1337.8  6355.3 1339.94  6405.1 1342.91  6435.7 1344.61
#Mann= 14 ,-1 , 0
  4139.4     .07       0  4154.5    .035       0  4747.2     .07       0
  4979.9     .05       0    5017     .07       0  5089.1     .07       0
  5139.7    .035       0  5344.6     .12       0  5472.4     .07       0
  5478.9     .12       0  5787.6     .07       0    6275     .12       0
  6355.3     .07       0  6405.1     .12       0
Bank Sta=4979.9,5017
XS Rating Curve= 0 ,0
Exp/Cntr=0.3,0.1

Type RM Length L Ch R = 1 ,59601   ,546,546,546
BEGIN DESCRIPTION:
CURRY CREEK 95.0
END DESCRIPTION:
XS GIS Cut Line= 3
        2105425.     13894324.98        2105475.       13893925.
      2104474.99     13892324.99
#Sta/Elev= 30
  4597.3  1305.4    4716 1302.85  4748.4 1299.36  4796.3 1286.88  4878.9 1279.59
    4950 1278.93  4980.2 1276.27  4989.5 1271.04  4990.5 1270.54  5026.6 1271.04
    5039 1273.26  5059.4 1276.65  5108.3 1277.48  5160.2  1284.9    5302 1288.06
  5449.1 1289.97  5522.2 1293.25  5824.1 1293.49  5894.1 1293.84  5942.4 1294.09
  6178.9 1296.32  6248.5 1297.06  6297.2 1298.34  6386.6  1297.9    6454 1300.05
  6459.4 1300.02  6648.4  1306.1  6721.5 1312.15  6769.9 1320.15  6887.2 1324.62
#Mann= 15 ,-1 , 0
  4597.3    .035       0    4716     .12       0  4878.9    .035       0
  4989.5    .035       0  5026.6    .035       0    5039     .12       0
    5302     .07       0  5824.1     .12       0  5894.1     .07       0
  5942.4     .12       0  6178.9     .07       0  6248.5     .12       0
  6297.2     .07       0    6454     .12       0  6459.4     .07       0
Bank Sta=4989.5,5026.6
XS Rating Curve= 0 ,0
Exp/Cntr=0.3,0.1

Type RM Length L Ch R = 1 ,59055   ,560,560,560
BEGIN DESCRIPTION:
CURRY CREEK 94.0
END DESCRIPTION:
XS GIS Cut Line= 3
      2106474.98     13894424.97        2105925.       13893675.
      2104484.37      13892095.4
#Sta/Elev= 30
  4074.5 1319.79  4124.1 1318.08  4196.8 1306.83  4414.5 1295.23    4646 1280.24
  4759.3    1284  4846.7  1285.8  4905.3 1284.15  4932.4 1280.79  4940.8 1276.69
  4978.6 1268.38  4979.6 1267.88  5015.7 1268.38  5018.4 1275.54  5082.5 1277.54
  5103.5 1283.54  5126.7 1284.98  5457.5 1284.31  5683.9 1291.18  5810.2 1290.13
  5960.2 1287.77  6139.1 1290.33  6211.4 1291.79    6413 1295.13  6866.2 1301.74
    6923 1306.13  6965.5 1311.16  6986.5 1316.96    7050 1323.33  7142.4 1326.97
#Mann= 10 ,-1 , 0
  4074.5     .07       0  4414.5    .035       0  4759.3     .12       0
  4978.6     .05       0  5015.7     .12       0  5126.7     .07       0
  5810.2     .12       0  6139.1     .07       0  6211.4     .12       0
    6413     .07       0
Bank Sta=4978.6,5015.7
XS Rating Curve= 0 ,0
Exp/Cntr=0.3,0.1
