HEC-RAS study CURRY CREEK.prj: CURRY CREEK Base Level Engineering

--- CURRY CREEK.g01 (geometry) --- (continued)

Type RM Length L Ch R = 1 ,28129   ,1630,1630,1630
BEGIN DESCRIPTION:
CURRY CREEK 45.0
END DESCRIPTION:
XS GIS Cut Line= 3
      2122474.98     13882124.96        2122125.       13881325.
      2120525.02     13880025.01
#Sta/Elev= 30
  4122.4  1192.9  4155.2 1191.09    4189 1189.54  4451.1 1178.97    4590 1175.64
  4887.6 1171.56  4962.4 1166.82  5002.4 1165.67  5023.6 1160.34  5066.7 1166.58
  5116.2 1163.63  5130.6 1165.23  5132.5 1160.04  5133.6 1159.44  5186.3 1160.04
  5188.1 1165.65  5223.3 1172.18  5769.7 1171.23  6080.9 1168.78  6365.2  1166.7
  6405.1 1166.15  6489.1 1166.89    6545 1171.14  6567.2 1176.27  6616.8 1200.64
    6652 1210.91  6773.4 1227.97  6828.9 1231.75  6954.1    1238  7057.1 1245.73
#Mann= 17 ,-1 , 0
  4122.4     .12       0  4155.2     .07       0    4189     .12       0
  4451.1    .035       0    4590     .07       0  4962.4     .12       0
  5002.4     .07       0  5132.5     .05       0  5186.3     .07       0
  5769.7    .035       0  6080.9     .07       0  6365.2    .035       0
  6405.1     .07       0  6489.1    .035       0  6567.2     .12       0
  6828.9     .07       0  6954.1     .12       0
Bank Sta=5132.5,5186.3
XS Rating Curve= 0 ,0
Exp/Cntr=0.3,0.1

Type RM Length L Ch R = 1 ,26499   ,550,550,550
BEGIN DESCRIPTION:
CURRY CREEK 44.0
END DESCRIPTION:
XS GIS Cut Line= 3
      2122524.99     13882075.04        2122925.       13880525.
        2122975.     13880125.03
#Sta/Elev= 30
  3394.8 1191.46  3414.5 1190.12  3514.2 1185.29  3611.3 1180.06    3782 1174.26
  4024.8 1168.75  4134.2 1168.36  4220.9 1164.35  4303.7 1164.98  4324.3 1163.74
  4337.6 1158.62  4355.3  1162.6  4378.2 1163.68  4427.6 1164.64  4458.8 1162.55
  4489.6 1160.46  4520.6 1163.88  4622.3 1164.27  4724.9 1162.64  4977.9 1160.21
  4978.3 1156.11  4979.5 1155.41    5033 1156.11  5033.4 1159.28    5046 1163.38
  5056.1 1174.01  5066.2  1176.3  5119.1 1180.13  5224.2 1182.71  5398.7 1188.48
#Mann= 12 ,-1 , 0
  3394.8     .12       0  3414.5     .07       0  3514.2     .12       0
  3611.3    .035       0    3782     .07       0  4220.9     .12       0
  4458.8    .035       0  4622.3     .12       0  4724.9     .07       0
  4978.3     .05       0    5033     .07       0  5224.2     .07       0
Bank Sta=4978.3,5033
XS Rating Curve= 0 ,0
Exp/Cntr=0.3,0.1

Type RM Length L Ch R = 1 ,25949   ,546,546,546
BEGIN DESCRIPTION:
CURRY CREEK 43.0
END DESCRIPTION:
XS GIS Cut Line= 3
      2122913.44     13882394.91        2123425.       13880675.
        2123375.     13880274.99
#Sta/Elev= 30
  3205.5 1199.93    3309 1194.69  3328.2 1194.22  3622.7 1181.53  3671.8 1177.73
  3803.3 1173.67  4290.4 1165.06  4362.5 1161.46  4426.2 1160.43  4446.9 1157.28
  4478.2  1160.5  4499.1 1155.55    4520  1160.5  4551.3  1161.2  4572.1 1158.09
  4597.6 1160.76  4662.6 1157.26  4707.8 1159.99  4764.3 1159.12  4822.5 1155.62
  4906.8 1157.27  4914.2 1157.45  5010.3 1154.18  5011.5 1153.48    5065 1154.18
  5080.5 1164.63  5091.7 1168.62    5151 1174.62  5354.4 1180.96    5403 1182.56
#Mann= 15 ,-1 , 0
  3205.5     .12       0    3309     .07       0  3328.2     .12       0
  3671.8    .035       0  3803.3     .07       0  4362.5     .12       0
  4597.6    .035       0  4662.6     .12       0  4764.3    .035       0
  4906.8     .07       0  4914.2    .035       0  5010.3    .035       0
    5065    .035       0  5091.7     .12       0  5354.4    .035       0
Bank Sta=5010.3,5065
XS Rating Curve= 0 ,0
Exp/Cntr=0.3,0.1

Type RM Length L Ch R = 1 ,25403   ,185,185,185
BEGIN DESCRIPTION:
CURRY CREEK 42.0
END DESCRIPTION:
XS GIS Cut Line= 3
      2123363.47     13882561.55        2123875.       13880875.
        2123825.     13880475.03
#Sta/Elev= 30
  3237.6  1190.2  3566.7 1183.63  3836.6 1171.58    3937  1168.7    4606 1160.17
    4697 1154.93  4717.9 1157.05  4742.8 1154.61  4780.9 1156.89  4801.5  1152.2
  4808.6 1154.65  4813.8 1153.08  4836.4 1156.38  4874.4 1154.42  4879.6  1156.2
  4895.5 1153.36  4950.7 1154.83  4958.2 1153.95  4962.2 1147.55  4963.4 1146.85
  5016.9 1147.55  5020.2 1152.42  5080.6 1151.98  5151.2 1154.84  5171.3 1150.98
  5204.1 1152.95  5211.7  1154.5  5231.8 1165.84    5252 1170.62  5403.1 1175.35
#Mann= 6 ,-1 , 0
  3237.6     .12       0  3836.6    .035       0    3937     .07       0
  4836.4     .12       0  4962.2     .05       0  5016.9     .12       0
Bank Sta=4962.2,5016.9
XS Rating Curve= 0 ,0
Exp/Cntr=0.3,0.1

Type RM Length L Ch R = 1 ,25218   ,391,391,391
BEGIN DESCRIPTION:
CURRY CREEK 41.5
END DESCRIPTION:
XS GIS Cut Line= 4
      2123822.89     13882563.52      2123975.04     13881445.95
      2124059.78     13880874.48      2123909.56     13880443.19
#Sta/Elev= 30
  3294.4 1186.91  3425.2 1182.75  3492.5 1177.02  3567.1 1172.87  3665.9 1169.04
  4014.4 1162.13  4198.4 1161.44  4199.8 1161.38    4358 1160.26  4456.9 1159.73
  4535.9 1159.21  4645.6 1159.25  4695.4 1156.26  4799.7 1152.93  4807.4 1154.46
  4869.1 1154.37  4989.4 1149.56  4993.2 1145.79  4994.4 1145.09    5048 1145.79
  5058.9 1149.71    5090 1151.78  5121.1 1152.46  5146.9 1150.49  5221.8 1153.86
  5240.1 1156.13  5302.3 1168.31  5370.1 1171.91    5426  1173.2  5456.7 1174.03
#Mann= 13 ,-1 , 0
  3294.4     .07       0  3567.1     .12       0  3665.9    .035       0
  4198.4     .07       0  4199.8    .035       0    4358     .07       0
  4456.9    .035       0  4535.9     .07       0  4695.4     .12       0
  4993.2     .05       0    5048     .12       0  5370.1    .035       0
    5426     .12       0
Bank Sta=4993.2,5048
XS Rating Curve= 0 ,0
Exp/Cntr=0.3,0.1

Type RM Length L Ch R = 1 ,24827   ,586,586,586
BEGIN DESCRIPTION:
CURRY CREEK 41.0
END DESCRIPTION:
XS GIS Cut Line= 3
      2124681.84     13882376.43        2124375.       13880675.
      2124024.99       13880475.
#Sta/Elev= 30
  3271.1 1176.76  3429.4 1172.81  3521.2 1169.82  3626.5 1165.05  3648.5 1165.74
  3732.4 1162.82  3858.6 1158.59  3891.3 1157.93  4070.3 1156.61    4235 1157.72
  4335.5 1158.06  4375.2 1157.34  4552.9 1155.91  4611.5 1153.33  4928.9 1148.97
  4979.7 1140.35  4980.5 1127.88  4981.7 1127.18  5035.3 1127.88  5045.3  1143.5
  5057.6 1147.43  5076.2 1149.29  5081.5 1149.56  5187.8 1154.23  5206.6 1155.08
  5233.9 1159.69  5314.6 1163.81  5330.4  1168.1  5345.5 1169.58  5403.1  1171.4
#Mann= 16 ,-1 , 0
  3271.1     .12       0  3429.4    .035       0  3521.2     .12       0
  3626.5    .035       0  3732.4     .07       0  3858.6    .035       0
  3891.3     .07       0    4235    .035       0  4335.5     .07       0
  4375.2    .035       0  4611.5     .12       0  4980.5     .05       0
  5035.3     .12       0  5076.2    .035       0  5081.5     .12       0
  5187.8    .035       0
Bank Sta=4980.5,5035.3
XS Rating Curve= 0 ,0
Exp/Cntr=0.3,0.1

Type RM Length L Ch R = 1 ,24241   ,570,570,570
BEGIN DESCRIPTION:
CURRY CREEK 40.0
END DESCRIPTION:
XS GIS Cut Line= 3
      2127309.51     13882092.98        2124775.       13880275.
      2124425.01     13880075.01
#Sta/Elev= 30
  1885.4 1195.03  2030.1 1188.83  2044.9 1185.24  2080.5 1185.88  2095.2 1181.63
  2195.9 1175.05  2338.4 1174.67  2432.4 1167.67  2631.3 1165.01  2717.8 1165.68
  2833.3 1157.69  3009.6 1157.72  3535.1 1152.47  3736.9 1149.33  4269.3 1152.42
  4534.9 1152.56  4665.7 1151.07  4825.2 1141.87  4875.6 1145.78  4915.2  1144.7
  4955.3 1141.58  4967.7 1136.23  4969.7 1128.31  4970.9 1127.61  5024.5 1128.31
  5027.5  1134.6  5055.6 1143.01  5098.1 1148.27  5216.1 1151.72  5407.6 1159.82
#Mann= 12 ,-1 , 0
  1885.4     .12       0  2631.3     .07       0  3009.6    .035       0
  3535.1     .12       0  4269.3    .035       0  4534.9     .07       0
  4665.7     .12       0  4915.2     .07       0  4969.7     .05       0
  5024.5     .07       0  5098.1     .12       0  5216.1    .035       0
#XS Ineff= 2 , 0
       0 4384.33 1155.93               0
Permanent Ineff=
       F       F
Bank Sta=4969.7,5024.5
XS Rating Curve= 0 ,0
Exp/Cntr=0.3,0.1

Type RM Length L Ch R = 1 ,24155   ,159,159,159
BEGIN DESCRIPTION:
CURRY CREEK 39.2
END DESCRIPTION:
XS GIS Cut Line= 3
      2127428.99     13881973.25      2124836.07     13880214.66
      2124476.33     13880022.44
#Sta/Elev= 30
  1866.3 1198.96  1995.9  1194.9  2071.1 1191.95  2112.8 1189.73  2156.1 1179.89
  2177.1  1186.1    2234 1189.32  2314.8  1179.4  2371.7  1181.8  2644.1 1176.01
    2803 1174.43  2900.9 1161.37  2925.1 1159.06  3080.5 1156.12    3625 1151.17
  4291.6 1152.41  4503.4 1153.38  4732.9 1148.53  4833.5 1141.42  4914.3 1145.13
    4963 1140.21  4992.2 1135.69  4995.8 1125.88    4997 1125.18  5050.6 1125.88
  5051.6 1135.08  5067.9 1141.28  5145.9 1149.14  5222.3 1151.12  5407.2 1157.45
#Mann= 16 ,-1 , 0
  1866.3     .12       0  1995.9     .07       0  2071.1     .12       0
  2644.1     .07       0  2900.9     .12       0  2925.1     .07       0
  3080.5    .035       0    3625     .12       0  4291.6    .035       0
  4503.4     .07       0  4732.9     .12       0    4963     .07       0
  4995.8     .05       0  5050.6     .07       0  5145.9     .12       0
  5222.3    .035       0
Bank Sta=4995.8,5050.6
XS Rating Curve= 0 ,0
Exp/Cntr=0.3,0.1

Type RM Length L Ch R = 1 ,23996   ,325,325,325
BEGIN DESCRIPTION:
CURRY CREEK 39.1
END DESCRIPTION:
XS GIS Cut Line= 3
       2127506.5     13881692.76      2124925.45     13880090.19
       2124480.3     13879904.57
#Sta/Elev= 30
  1961.9 1201.83  2307.6  1195.5  2770.1 1191.25  2955.6 1170.73  3007.6 1157.49
  3074.7 1154.72  3092.1 1154.77  3188.5 1153.74  3288.3 1153.55  3416.2 1153.22
  3484.4 1152.35  3696.1 1147.85  4314.3  1151.9  4440.7 1152.57  4465.1 1152.34
  4662.1 1150.01  4821.9  1141.7  4939.6 1140.11  4945.5 1131.84  4953.4 1096.89
  4966.8 1103.93  4994.2 1093.75  4995.4 1093.05    5049 1093.75  5133.2 1102.43
  5151.6 1146.87  5157.4 1146.41  5207.6  1149.3  5451.3 1156.29  5482.3 1156.55
#Mann= 18 ,-1 , 0
  1961.9     .12       0  2307.6     .07       0  2770.1     .12       0
  3074.7     .07       0  3092.1     .12       0  3188.5    .035       0
  3288.3     .07       0  3416.2    .035       0  3484.4     .12       0
  4314.3    .035       0  4440.7     .12       0  4465.1     .07       0
  4821.9     .12       0  4994.2     .05       0    5049     .12       0
  5157.4     .12       0  5207.6    .035       0  5451.3     .07       0
Bank Sta=4994.2,5049
XS Rating Curve= 0 ,0
Exp/Cntr=0.3,0.1

Type RM Length L Ch R = 1 ,23671   ,563,563,563
BEGIN DESCRIPTION:
CURRY CREEK 39.0
END DESCRIPTION:
XS GIS Cut Line= 3
      2127045.83     13880930.35        2125075.       13879825.
      2124675.04       13879825.
#Sta/Elev= 30
  2740.6 1202.51    3009 1190.09  3127.7  1160.7  3169.8 1154.99  3360.7 1149.14
  3725.2 1147.07    3837  1146.5  3966.4  1146.3  4023.5 1147.74  4419.4 1151.26
  4752.1 1145.52  4802.8 1141.52  4808.5 1135.34  4816.8 1116.82  4824.5 1111.13
  4830.2 1111.92  4839.7 1104.11  4883.8  1096.1  4889.6 1088.65  4905.5 1097.11
  4947.2 1093.45  4970.6 1080.07  5012.8 1077.22    5014 1076.52  5067.6 1077.22
  5070.2 1081.66  5140.2 1105.06  5150.2 1145.14  5289.8 1148.88  5400.2 1150.45
#Mann= 11 ,-1 , 0
  2740.6     .12       0  3169.8     .07       0  3725.2     .12       0
    3837     .07       0  3966.4     .12       0  4023.5     .07       0
  4752.1     .12       0  4947.2     .07       0  5012.8     .05       0
  5067.6     .07       0  5289.8    .035       0
Bank Sta=5012.8,5067.6
XS Rating Curve= 0 ,0
Exp/Cntr=0.3,0.1

Type RM Length L Ch R = 1 ,23108   ,549,549,549
BEGIN DESCRIPTION:
CURRY CREEK 38.0
END DESCRIPTION:
XS GIS Cut Line= 3
      2127377.71     13880333.63        2125425.       13879425.
      2125024.98       13879375.
#Sta/Elev= 30
  2846.3 1205.27  3092.5  1195.1  3172.7 1191.67  3367.7 1157.36  3708.6    1139
  3820.9  1145.1  4065.9 1135.78  4083.3 1107.04  4102.3 1104.16  4194.9 1096.21
    4217 1109.93  4226.1 1128.57  4231.6 1109.02    4239  1131.4    4249 1136.45
  4368.9 1144.21    4784 1143.69  4878.7 1140.99  4888.8 1121.64  4894.3 1098.23
  4900.8 1092.58  4958.4 1076.79  4959.6 1076.09  5013.3 1076.79  5161.3 1086.45
  5192.9 1098.82  5231.9 1111.93    5252 1128.82  5291.8 1136.28  5403.2 1144.24
#Mann= 11 ,-1 , 0
  2846.3     .12       0  3092.5     .07       0  3172.7     .12       0
  3708.6     .07       0  3820.9     .12       0  4102.3     .07       0
    4784     .12       0  4958.4     .05       0  5013.3     .12       0
  5192.9     .12       0  5291.8     .12       0
#XS Ineff= 2 , 0
       0 4309.66 1139.67               0
Permanent Ineff=
       F       F
Bank Sta=4958.4,5013.3
XS Rating Curve= 0 ,0
Exp/Cntr=0.3,0.1

Type RM Length L Ch R = 1 ,22559   ,582,582,582
BEGIN DESCRIPTION:
CURRY CREEK 37.0
END DESCRIPTION:
XS GIS Cut Line= 3
      2125774.97     13878625.03        2125475.       13878925.
      2125125.03     13879124.98
#Sta/Elev= 30
  4576.4 1150.74  4632.9 1147.72  4647.1 1139.67  4661.2 1127.17  4675.4 1119.97
  4689.5 1114.35  4717.8 1112.18  4731.9 1098.52  4736.4 1096.37  4746.1 1091.74
  4774.4 1085.34  4788.5 1083.87  4816.8 1076.38  4932.7 1077.97  4986.5 1077.96
  4996.2 1075.53  4997.4 1074.83  5051.1 1075.53  5051.7 1077.28  5061.7    1078
  5112.5 1084.25  5132.4 1083.01  5184.9 1091.78  5219.5 1105.37  5234.6 1108.22
  5250.4 1114.11  5265.5 1132.93    5272 1134.37  5352.6 1141.07  5403.7 1141.62
#Mann= 7 ,-1 , 0
  4576.4     .12       0  4736.4     .12       0  4932.7     .12       0
  4996.2     .05       0  5051.1     .12       0  5061.7     .12       0
  5112.5     .12       0
Bank Sta=4996.2,5051.1
XS Rating Curve= 0 ,0
Exp/Cntr=0.3,0.1

Type RM Length L Ch R = 1 ,21977   ,567,567,567
BEGIN DESCRIPTION:
CURRY CREEK 36.0
END DESCRIPTION:
XS GIS Cut Line= 3
        2125625.       13878475.        2125225.       13878475.
        2125175.     13878874.99
#Sta/Elev= 30
  4600.5 1146.57  4740.5 1139.23  4750.5 1132.83  4760.5 1100.63  4790.5  1088.2
  4840.5 1081.53  4880.5 1072.56  4890.5 1072.34  4920.5 1076.52  4970.5 1077.48
  4980.5 1075.26  4982.4 1070.63  4983.7 1069.83  5038.8 1070.63  5043.3 1079.77
  5091.2  1075.9  5101.3  1073.2  5131.5 1075.33  5151.7 1073.68  5161.7 1074.34
  5181.9 1078.51  5204.6 1086.05  5212.1 1086.05  5232.3 1094.63  5262.5  1101.3
  5285.2 1110.59  5302.8 1121.27  5312.9 1125.43    5323 1132.48  5403.6 1134.95
#Mann= 3 ,-1 , 0
  4600.5     .12       0  4982.4     .05       0  5038.8     .12       0
Bank Sta=4982.4,5038.8
XS Rating Curve= 0 ,0
Exp/Cntr=0.3,0.1

Type RM Length L Ch R = 1 ,21410   ,553,553,553
BEGIN DESCRIPTION:
CURRY CREEK 35.0
END DESCRIPTION:
XS GIS Cut Line= 3
      2125074.99       13878075.        2124725.       13878275.
        2124625.     13878674.99
#Sta/Elev= 30
  4602.9 1138.92  4691.4 1137.34  4728.9 1132.82  4772.1 1119.42  4777.8 1111.89
  4793.7 1107.72  4799.4    1101  4809.5 1099.59  4815.2 1094.26  4831.1 1089.34
  4836.8 1084.68  4852.7  1081.1  4858.4 1076.96  4890.1 1072.26  4960.7 1073.97
  4964.1 1066.23  4965.4 1065.43  5020.5 1066.23    5024 1073.54  5029.2  1074.5
  5070.4  1074.6  5088.5 1070.02  5106.5 1069.19  5170.9 1082.15  5222.5 1088.13
  5317.8 1111.99  5325.5 1116.12  5366.8 1129.09  5387.4 1132.92  5418.3 1134.14
#Mann= 3 ,-1 , 0
  4602.9     .12       0  4964.1     .05       0  5020.5     .12       0
Bank Sta=4964.1,5020.5
XS Rating Curve= 0 ,0
Exp/Cntr=0.3,0.1

Type RM Length L Ch R = 1 ,20857   ,539,539,539
BEGIN DESCRIPTION:
CURRY CREEK 34.0
END DESCRIPTION:
XS GIS Cut Line= 3
        2124425.       13877775.        2124225.       13878125.
      2123875.02     13878324.99
#Sta/Elev= 30
    4596 1130.67  4676.6 1127.31  4743.6 1116.78  4780.3 1101.27  4792.5  1093.8
  4824.2 1079.52  4845.8 1072.89    4889  1070.8  4918.5 1066.74  4941.5 1068.81
  4963.8 1063.75  4999.1 1064.91  5000.4 1062.37  5001.7 1061.57  5056.9 1062.37
  5066.1 1070.42  5071.8 1073.36  5093.4 1078.96  5125.1 1078.47  5130.8 1081.91
  5146.7 1084.63    5174 1092.71  5217.9 1100.38  5233.1 1105.34    5241 1124.37
  5248.9 1130.77  5254.7 1128.64  5272.7 1132.18  5278.7  1132.5  5402.2 1138.03
#Mann= 5 ,-1 , 0
    4596     .12       0  5000.4     .05       0  5056.9     .12       0
  5272.7     .07       0  5278.7    .035       0
Bank Sta=5000.4,5056.9
XS Rating Curve= 0 ,0
Exp/Cntr=0.3,0.1

Type RM Length L Ch R = 1 ,20318   ,556,556,556
BEGIN DESCRIPTION:
CURRY CREEK 33.0
END DESCRIPTION:
XS GIS Cut Line= 3
      2124224.96     13877575.02        2123875.       13877775.
      2123474.98       13877825.
#Sta/Elev= 30
  4596.6 1130.33  4631.8 1126.45  4647.7 1120.94  4654.1 1116.51  4706.7 1095.55
  4728.3 1090.22  4734.8 1087.45  4824.7 1077.55  4942.1 1068.98  4948.6 1066.48
  4970.1 1065.37  4991.6 1060.92  4992.8 1060.12  5048.1 1060.92  5050.1 1069.95
  5060.1 1071.99  5080.3 1073.12  5090.4 1075.96  5107.7 1083.24  5118.1 1087.71
  5123.1 1087.86  5140.8 1092.56    5171 1102.62  5191.1 1112.58  5211.3 1125.75
  5231.5 1131.84  5269.6 1136.99  5322.2 1141.43  5359.9 1146.62  5402.8 1149.71
#Mann= 5 ,-1 , 0
  4596.6     .12       0  4991.6     .05       0  5048.1     .12       0
  5107.7     .07       0  5269.6    .035       0
Bank Sta=4991.6,5048.1
XS Rating Curve= 0 ,0
Exp/Cntr=0.3,0.1

Type RM Length L Ch R = 1 ,19762   ,543,543,543
BEGIN DESCRIPTION:
CURRY CREEK 32.0
END DESCRIPTION:
XS GIS Cut Line= 3
      2124274.98     13877474.99        2123925.       13877275.
        2123725.     13876925.01
#Sta/Elev= 30
  4597.3 1131.98  4735.5 1129.75  4781.6 1119.97    4788 1116.03  4809.6 1110.91
  4847.1 1094.25  4906.1 1076.43  4970.9 1066.94  4977.4 1061.68  5001.5 1055.79
  5002.8 1054.99  5058.3 1055.79  5073.1 1061.47  5088.9 1062.13  5110.5 1058.28
    5148 1067.86  5153.7 1072.33  5169.6 1074.31  5175.3 1079.13  5184.7 1081.88
  5196.9 1091.55  5212.7 1096.81  5228.6 1098.07  5250.2 1105.54  5255.9 1131.79
  5265.3 1143.74  5277.5 1154.23  5293.4 1155.77  5336.6 1175.28  5403.5 1187.44
#Mann= 3 ,-1 , 0
  4597.3     .12       0  5001.5     .05       0  5058.3     .12       0
Bank Sta=5001.5,5058.3
XS Rating Curve= 0 ,0
Exp/Cntr=0.3,0.1

Type RM Length L Ch R = 1 ,19219   ,550,550,550
BEGIN DESCRIPTION:
CURRY CREEK 31.0
END DESCRIPTION:
XS GIS Cut Line= 3
        2124225.     13877324.99        2124275.       13876925.
        2124225.     13876525.02
#Sta/Elev= 30
  4601.8 1123.15  4621.9 1120.38  4672.3 1107.27  4732.8 1088.72  4773.1 1084.23
  4800.8 1076.41    4894 1068.16  4914.2  1062.7  4954.5 1062.56  4962.1 1059.45
  4967.1 1060.49    4974 1055.56  4975.3 1054.76  5030.8 1055.56  5042.7 1068.15
  5047.7 1068.62  5055.3 1078.06  5115.8 1109.45  5123.3 1125.95  5128.4 1130.41
  5135.9 1140.94  5156.1 1154.71  5176.2 1159.39  5203.9 1175.28    5209 1175.27
  5216.5 1180.23  5246.8 1191.73  5266.9 1195.03    5319 1197.72    5408 1201.78
#Mann= 4 ,-1 , 0
  4601.8     .12       0    4974     .05       0  5030.8     .12       0
    5319     .07       0
Bank Sta=4974,5030.8
XS Rating Curve= 0 ,0
Exp/Cntr=0.3,0.1

Type RM Length L Ch R = 1 ,18669   ,579,579,579
BEGIN DESCRIPTION:
CURRY CREEK 30.0
END DESCRIPTION:
XS GIS Cut Line= 3
        2124825.       13877475.        2124775.       13877075.
        2124775.     13876675.01
#Sta/Elev= 30
  4602.3 1133.19  4682.9 1129.92  4713.2 1121.28  4720.7 1116.29  4725.8  1115.8
  4801.3 1083.38  4806.4 1083.96  4813.9  1080.2  4834.1 1075.61    4887 1072.67
  4914.7 1067.74  4924.8 1065.04  4944.9 1054.35  4956.9  1054.3  4958.2  1053.5
  5013.7  1054.3  5015.4 1056.15  5035.4 1062.77  5055.4 1066.24  5065.4  1071.7
  5095.4  1078.1  5135.4 1104.66  5145.4 1114.19  5155.4 1126.19  5165.4 1145.22
  5185.4 1153.82  5215.4 1158.83  5265.4 1176.77  5329.7 1189.79  5405.4 1192.77
#Mann= 4 ,-1 , 0
  4602.3     .12       0  4956.9     .05       0  5013.7     .12       0
  5329.7    .035       0
Bank Sta=4956.9,5013.7
XS Rating Curve= 0 ,0
Exp/Cntr=0.3,0.1

Type RM Length L Ch R = 1 ,18090   ,556,556,556
BEGIN DESCRIPTION:
CURRY CREEK 29.0
END DESCRIPTION:
XS GIS Cut Line= 3
        2125325.     13877575.04        2125325.       13877175.
      2125124.98     13876824.96
#Sta/Elev= 30
  4595.8 1135.05  4755.8 1130.83  4805.8 1127.23  4825.8  1120.7  4905.8 1088.07
  4925.8 1077.52  4935.8 1076.61  4955.8 1068.82  4965.8  1067.4  4975.3  1053.5
  4976.6  1052.7  5032.2  1053.5  5041.2 1059.11  5062.8 1061.63  5127.6 1063.42
  5170.8 1068.67  5186.6  1075.6  5208.2 1079.74    5224 1086.46  5229.8 1086.93
  5288.8 1110.31  5304.7 1118.99  5310.4 1119.46  5318.3 1125.35  5326.3 1137.98
    5332 1138.76  5341.4 1148.95  5347.8 1151.61  5363.7 1154.91    5399 1157.16
#Mann= 3 ,-1 , 0
  4595.8     .12       0  4975.3     .05       0  5032.2     .12       0
Bank Sta=4975.3,5032.2
XS Rating Curve= 0 ,0
Exp/Cntr=0.3,0.1

Type RM Length L Ch R = 1 ,17534   ,717,717,717
BEGIN DESCRIPTION:
CURRY CREEK 28.0
END DESCRIPTION:
XS GIS Cut Line= 3
        2125625.       13877425.        2125825.       13877075.
      2125352.51     13876378.93
#Sta/Elev= 30
  4592.9 1127.67  4696.6 1115.76  4762.1 1092.02  4821.1 1076.48    4990 1053.85
  4991.3 1053.05  5046.9 1053.85  5054.4 1056.14  5075.4 1055.89  5132.3 1062.05
  5147.2 1068.93  5168.2 1071.91  5189.4 1078.66  5219.1 1082.22    5234 1087.12
    5255 1091.05  5284.9 1102.59    5291 1102.74  5305.9 1113.42  5326.9 1119.99
  5341.8 1130.59    5402 1136.59  5523.5  1142.9  5546.2 1144.55  5572.4 1144.09
  5593.4 1147.06  5614.4  1147.5  5623.3 1145.89  5737.1 1151.28  5837.3 1151.62
#Mann= 6 ,-1 , 0
  4592.9     .12       0    4990     .05       0  5046.9     .12       0
    5402     .07       0  5523.5    .035       0  5546.2     .07       0
Bank Sta=4990,5046.9
XS Rating Curve= 0 ,0
Exp/Cntr=0.3,0.1

Type RM Length L Ch R = 1 ,16817   ,380,380,380
BEGIN DESCRIPTION:
CURRY CREEK 27.0
END DESCRIPTION:
XS GIS Cut Line= 3
        2126475.     13877324.97      2126414.33     13876930.02
      2126148.69     13876122.68
#Sta/Elev= 30
  4606.6 1124.97  4657.2 1118.24    4704 1103.17  4709.1  1105.8    4728 1096.98
  4748.2 1091.02  4854.2 1067.36  4879.7 1059.12  4960.7 1051.18  4972.5 1047.97
  4973.9 1047.17  5029.7 1047.97  5032.5  1054.9  5150.8 1078.95  5177.3 1087.58
  5182.6 1086.65  5209.1 1096.72  5214.4 1095.11  5240.9 1104.78  5246.2 1103.27
  5272.7  1108.9    5278 1106.97  5304.5 1114.65  5309.7 1111.73  5336.3 1117.87
  5341.5 1115.22  5368.1 1120.98  5500.5 1122.05  5640.6 1129.74  5856.1 1136.16
#Mann= 5 ,-1 , 0
  4606.6     .12       0  4854.2    .035       0  4972.5     .05       0
  5029.7    .035       0  5640.6     .07       0
Bank Sta=4972.5,5029.7
XS Rating Curve= 0 ,0
Exp/Cntr=0.3,0.1

Type RM Length L Ch R = 1 ,16437   ,519,519,519
BEGIN DESCRIPTION:
CURRY CREEK 26.0
END DESCRIPTION:
XS GIS Cut Line= 3
        2126975.       13877225.        2126775.       13876875.
      2126575.01     13876525.02
#Sta/Elev= 30
  4601.5  1131.4  4682.1 1125.57  4705.2 1120.09  4711.6 1115.58  4749.1 1098.26
  4754.8 1097.75  4770.7  1088.2  4776.4 1088.29  4792.3  1081.5    4798 1082.64
  4813.9 1079.27  4820.3 1075.04  4835.4 1073.88    4857 1068.26  4872.9 1061.44
  4959.3  1052.4  4968.1 1048.09  4969.4 1047.29  5025.3 1048.09  5027.6 1053.63
  5034.1 1055.26  5098.9 1063.27  5114.7 1068.17  5136.3 1070.49  5165.9 1076.98
    5217 1092.58  5232.8 1101.53    5276 1114.61  5313.4 1119.37  5407.7 1123.62
#Mann= 3 ,-1 , 0
  4601.5     .12       0  4968.1     .05       0  5025.3     .12       0
Bank Sta=4968.1,5025.3
XS Rating Curve= 0 ,0
Exp/Cntr=0.3,0.1

Type RM Length L Ch R = 1 ,15918   ,542,542,542
BEGIN DESCRIPTION:
CURRY CREEK 25.0
END DESCRIPTION:
XS GIS Cut Line= 3
      2127425.01     13877025.02        2127225.       13876675.
      2126874.96     13876424.97
#Sta/Elev= 30
  4596.9 1132.22    4648 1130.03  4700.6 1123.81  4707.1 1120.86  4712.8 1120.21
  4744.5 1106.27  4750.3 1105.04  4766.1 1096.35  4781.2 1090.71  4793.4 1084.25
  4803.5    1081  4809.3 1083.01  4838.8 1078.37  4874.1 1060.33  4919.4 1054.44
  4920.3 1048.17  4921.6 1047.37  4977.5 1048.17  5003.1 1050.87  5013.6 1056.08
  5022.2 1057.11  5063.9 1056.95  5149.2 1062.78  5158.1 1064.13  5229.8 1076.16
  5250.7 1081.53  5307.3 1099.95  5336.8  1106.1    5408 1116.19  5430.2 1117.99
#Mann= 5 ,-1 , 0
  4596.9     .12       0  4920.3     .05       0  4977.5     .12       0
  5149.2     .07       0  5158.1     .12       0
Bank Sta=4920.3,4977.5
XS Rating Curve= 0 ,0
Exp/Cntr=0.3,0.1

Type RM Length L Ch R = 1 ,15376   ,532,532,532
BEGIN DESCRIPTION:
CURRY CREEK 24.0
END DESCRIPTION:
XS GIS Cut Line= 3
      2127875.03       13876225.        2127475.       13876225.
      2126975.03       13876175.
#Sta/Elev= 30
  4595.6 1126.68  4643.5 1124.61  4685.6 1121.92  4715.6 1116.11  4735.6 1114.44
  4785.6 1103.52  4815.6 1090.48  4835.6 1083.58  4875.6 1073.38  4895.6 1065.89
  4905.6 1059.34  4915.6    1055  4965.6 1051.51  4993.1 1047.73  5025.8 1047.54
  5027.3 1045.65  5028.6 1044.85  5084.6 1045.65  5086.1 1048.79  5106.2 1052.81
  5126.3 1059.58    5169 1062.72  5256.9 1072.55    5277 1077.36  5297.1 1079.05
  5349.9 1091.14  5397.6 1104.36  5450.4 1112.44    5468 1116.85  5498.1 1118.22
#Mann= 5 ,-1 , 0
  4595.6     .07       0  4643.5     .12       0  5027.3     .05       0
  5084.6     .12       0    5169     .12       0
Bank Sta=5027.3,5084.6
XS Rating Curve= 0 ,0
Exp/Cntr=0.3,0.1

Type RM Length L Ch R = 1 ,14844   ,554,554,554
BEGIN DESCRIPTION:
CURRY CREEK 23.0
END DESCRIPTION:
XS GIS Cut Line= 3
      2127724.98     13875924.99        2127375.       13875725.
      2126389.16     13875961.06
#Sta/Elev= 30
  4596.5 1121.38  4647.6 1116.63  4690.8 1103.33  4706.6 1092.64  4749.8 1081.32
  4765.6 1071.06  4808.8 1067.83  4815.3 1055.95  4824.7 1051.65  4830.4 1056.22
  4846.3 1048.46  4889.5 1047.35  4905.3 1041.85    4963 1040.89  4964.4 1040.09
  5020.3 1040.89  5023.2 1050.36  5040.7 1057.94  5275.4 1076.57    5380 1101.24
  5453.8 1104.78  5532.8 1100.34  5627.1 1102.49    5664 1095.19  5739.9 1088.64
  5770.8 1093.81  5790.1 1102.96  5842.8  1116.1  6001.3 1131.09  6013.3 1131.76
#Mann= 4 ,-1 , 0
  4596.5     .12       0    4963     .05       0  5020.3     .12       0
  6001.3     .07       0
Bank Sta=4963,5020.3
XS Rating Curve= 0 ,0
Exp/Cntr=0.3,0.1

Type RM Length L Ch R = 1 ,14290   ,538,538,538
BEGIN DESCRIPTION:
CURRY CREEK 22.0
END DESCRIPTION:
XS GIS Cut Line= 3
      2127724.97     13875624.97        2127425.       13875225.
      2126732.06     13874445.67
#Sta/Elev= 30
  4500.1  1107.6  4503.9 1107.55  4557.3  1100.6  4600.1 1086.47  4642.8 1076.98
  4674.6 1073.83  4753.6 1065.96  4832.4 1061.78  4906.3 1055.11  4942.8 1043.68
  4978.2 1040.77  4978.4 1038.79  4979.7 1037.99    5036 1038.79  5070.7 1041.01
  5113.4 1047.76  5120.5 1046.69  5127.6 1049.57  5134.3 1060.25  5191.1 1079.04
    5248 1092.22  5319.1 1116.53  5449.3 1128.17  5615.9  1137.8  5651.9 1144.45
  5708.7 1148.66  5821.6 1154.47  5892.7 1169.77  5970.5 1175.43  6042.9 1175.89
#Mann= 9 ,-1 , 0
  4500.1     .07       0  4503.9     .12       0  4600.1     .07       0
  4674.6     .12       0  4753.6     .07       0  4832.4     .12       0
  4978.4     .05       0    5036     .12       0  5449.3     .07       0
Bank Sta=4978.4,5036
XS Rating Curve= 0 ,0
Exp/Cntr=0.3,0.1

Type RM Length L Ch R = 1 ,13752   ,540,540,540
BEGIN DESCRIPTION:
CURRY CREEK 21.0
END DESCRIPTION:
XS GIS Cut Line= 3
        2127875.     13875675.02        2127775.       13874875.
      2127424.96     13874674.98
#Sta/Elev= 30
  4193.1 1117.92  4225.1 1115.63  4263.7 1108.97  4324.4 1101.57  4364.4 1095.57
  4561.9 1077.48  4738.2 1067.03  4777.6  1063.9  4837.7 1056.35  4937.2 1045.03
    4949 1043.85  4950.4  1036.1  4951.7  1035.3    5008  1036.1    5013 1039.21
  5022.4 1039.98  5028.9 1042.44  5034.6  1048.3  5044.7 1049.71  5050.5 1058.88
  5066.3 1059.68    5080 1062.77  5109.5 1072.39  5160.6 1085.89  5168.5 1086.63
  5211.7 1100.02  5249.9 1116.06  5264.2 1119.02  5298.8 1121.84  5402.5  1127.1
#Mann= 10 ,-1 , 0
  4193.1     .07       0  4225.1     .12       0  4324.4     .07       0
  4561.9     .12       0  4738.2     .07       0  4837.7    .035       0
  4937.2     .12       0  4950.4     .05       0    5008     .12       0
  5249.9     .07       0
Bank Sta=4950.4,5008
XS Rating Curve= 0 ,0
Exp/Cntr=0.3,0.1

Type RM Length L Ch R = 1 ,13212   ,539,539,539
BEGIN DESCRIPTION:
CURRY CREEK 20.0
END DESCRIPTION:
XS GIS Cut Line= 3
        2128225.       13875525.        2128275.       13874825.
        2128475.       13874475.
#Sta/Elev= 30
  4298.1 1114.27  4418.4 1099.42  4448.5 1094.47  4558.8 1082.23  4839.5 1056.18
  4873.1 1054.55  4909.7 1049.42  4927.2 1043.85  4968.5 1036.58  4969.9 1035.68
  5026.2 1036.58  5029.4 1045.92  5057.5 1046.89  5066.8 1059.68  5072.6 1059.97
  5088.4 1065.02  5094.2 1065.51    5110  1071.1  5125.9 1072.61  5131.6 1071.26
    5169 1087.69  5174.8  1087.4  5190.6 1095.15  5196.4 1095.36  5206.5 1099.71
  5228.1 1113.89  5241.8 1121.53  5249.7 1124.35  5292.9  1129.9    5403 1135.28
#Mann= 4 ,-1 , 0
  4298.1     .07       0  4873.1     .12       0  4968.5     .05       0
  5026.2     .12       0
Bank Sta=4968.5,5026.2
XS Rating Curve= 0 ,0
Exp/Cntr=0.3,0.1

Type RM Length L Ch R = 1 ,12673   ,549,549,549
BEGIN DESCRIPTION:
CURRY CREEK 19.0
END DESCRIPTION:
XS GIS Cut Line= 3
      2128539.33     13875956.07        2128725.       13875075.
        2128725.     13874675.02
#Sta/Elev= 30
  4095.3 1122.09  4207.9 1120.88  4251.4 1120.07  4438.4  1116.6  4488.7 1111.66
  4587.8    1102    4609  1095.8  4677.2 1079.42  4726.9 1071.23  4801.5 1063.78
  4944.6 1054.64  4965.1 1048.78  4970.8 1044.04  4975.9 1044.42  4993.2 1037.02
  5006.9 1035.68  5016.9 1035.55  5018.2 1034.65  5074.6 1035.55  5095.7 1044.02
  5105.7 1045.74  5135.7 1059.51  5195.7 1075.43  5235.7 1089.42  5265.7 1103.26
  5275.7 1109.88  5285.7 1120.81  5295.7 1125.81  5315.7 1128.27  5395.7 1131.33
#Mann= 8 ,-1 , 0
  4095.3    .035       0  4207.9     .07       0  4251.4     .12       0
  4488.7     .07       0    4609    .035       0  5006.9     .12       0
  5016.9    .035       0  5074.6     .12       0
Bank Sta=5016.9,5074.6
XS Rating Curve= 0 ,0
Exp/Cntr=0.3,0.1

Type RM Length L Ch R = 1 ,12124   ,586,586,586
BEGIN DESCRIPTION:
CURRY CREEK 18.0
END DESCRIPTION:
XS GIS Cut Line= 3
      2129299.75     13875982.12        2129225.       13875225.
      2129124.99     13874774.98
#Sta/Elev= 30
  4243.8 1125.68  4351.4 1121.87  4401.7 1117.26  4445.9 1116.35    4542 1106.49
  4556.7 1103.34  4592.6 1097.23  4637.3 1083.56    4673 1074.18  4855.4 1056.66
  4863.9 1053.05  4874.5 1045.52  4904.1 1043.35  4924.2 1038.09  4965.6  1035.7
    4967  1034.8  5023.5  1035.7  5023.8 1037.27  5045.6 1038.84    5116 1052.42
  5213.3 1062.35    5262 1069.65  5300.4 1079.69  5305.5 1079.33  5311.9 1082.63
  5342.6 1092.42  5349.1 1097.06  5354.2 1096.93  5414.4 1119.44  5465.6 1123.98
#Mann= 6 ,-1 , 0
  4243.8     .12       0  4556.7     .07       0  4637.3    .035       0
  4874.5     .12       0  4965.6     .05       0  5023.5     .12       0
Bank Sta=4965.6,5023.5
XS Rating Curve= 0 ,0
Exp/Cntr=0.3,0.1

Type RM Length L Ch R = 1 ,11538   ,578,578,578
BEGIN DESCRIPTION:
CURRY CREEK 17.0
END DESCRIPTION:
XS GIS Cut Line= 3
      2130174.98     13875574.99        2129775.       13875325.
        2129525.     13874674.99
#Sta/Elev= 30
  4528.4 1117.49  4557.3 1114.88  4563.7 1111.74  4636.3 1089.93  4724.7 1071.97
  4782.5 1064.53    4865 1056.47  4869.1 1056.33  4892.2 1054.67  4913.4 1051.22
  4919.3 1039.49  4928.7 1038.64    4950 1032.22  4980.7 1030.71  4982.1 1029.81
  5038.7 1030.71  5039.7 1036.23  5045.1 1036.24  5053.6 1040.23  5094.4  1046.6
  5124.4 1049.25    5239 1054.21  5323.6 1059.99  5402.9 1068.01  5432.9 1069.69
  5503.6 1078.64  5557.2 1087.59  5596.8 1100.03  5664.3 1113.81  5696.5 1115.81
#Mann= 5 ,-1 , 0
  4528.4     .12       0    4865     .07       0  4869.1     .12       0
  4980.7     .05       0  5038.7     .12       0
Bank Sta=4980.7,5038.7
XS Rating Curve= 0 ,0
Exp/Cntr=0.3,0.1

Type RM Length L Ch R = 1 ,10960   ,524,524,524
BEGIN DESCRIPTION:
CURRY CREEK 16.0
END DESCRIPTION:
XS GIS Cut Line= 3
      2130474.98     13875474.97        2130275.       13875125.
        2129925.     13874625.01
#Sta/Elev= 30
  4607.2 1128.97  4680.6 1126.02  4738.9  1122.7  4745.4 1116.33  4754.7 1111.96
  4760.5 1107.23  4768.4 1104.71  4776.3 1098.77  4791.4 1092.67  4797.9 1087.76
  4819.5  1080.9  4835.4 1072.26    4849 1067.87  4872.1 1065.33  4884.3  1058.6
  4894.4 1044.47  4906.6  1040.9  4908.6 1031.44  4909.9 1030.54  4966.6 1031.44
  4987.2    1032  5007.4 1040.59  5053.4 1047.25  5150.3 1053.11  5211.3 1054.48
    5273 1058.88  5348.1 1067.85  5491.1 1081.66  5592.3 1099.47  5620.6 1102.27
#Mann= 6 ,-1 , 0
  4607.2     .07       0  4680.6     .12       0  4908.6     .05       0
  4966.6     .12       0  5150.3    .035       0    5273     .12       0
Bank Sta=4908.6,4966.6
XS Rating Curve= 0 ,0
Exp/Cntr=0.3,0.1

Type RM Length L Ch R = 1 ,10436   ,686,686,686
BEGIN DESCRIPTION:
CURRY CREEK 15.0
END DESCRIPTION:
XS GIS Cut Line= 3
        2130725.       13875425.        2130725.       13875025.
      2130075.03     13874325.03
#Sta/Elev= 30
  4580.9 1123.62  4680.9  1121.5  4790.9 1116.55  4803.4 1114.61  4820.9 1110.79
  4853.2 1095.21  4870.9 1087.87  4880.9 1079.16  4890.9 1075.76  4900.9 1077.15
  4940.9 1061.41  4970.9 1055.38  4978.4 1041.07  4979.4 1041.07  4984.3 1041.07
  4994.1 1029.66  4995.5 1028.76  5052.1 1029.66  5058.8 1033.79  5087.2 1042.26
  5195.5 1049.22  5255.1 1052.04  5302.4 1052.98    5363 1054.45  5452.3  1060.1
  5490.3 1065.96  5592.5 1073.59  5732.7 1085.64  5807.8 1095.31  5936.1 1106.17
#Mann= 13 ,-1 , 0
  4580.9     .07       0  4803.4     .12       0  4853.2     .07       0
  4979.4     .12       0  4994.1     .05       0  5052.1     .12       0
  5195.5     .12       0  5255.1     .12       0  5302.4    .035       0
  5452.3     .12       0  5592.5    .035       0  5732.7     .12       0
  5807.8    .035       0
Bank Sta=4994.1,5052.1
XS Rating Curve= 0 ,0
Exp/Cntr=0.3,0.1

Type RM Length L Ch R = 1 ,9750    ,669,669,669
BEGIN DESCRIPTION:
CURRY CREEK 14.0
END DESCRIPTION:
XS GIS Cut Line= 3
      2131474.97       13874475.        2130975.       13874475.
      2130075.02     13874275.01
#Sta/Elev= 30
    4492 1123.57    4540 1120.34    4612 1114.42    4632 1109.81  4669.5 1097.03
    4732 1074.69    4752 1076.23    4772 1074.33    4782  1071.3    4802 1071.24
  4863.4 1060.32    4892 1055.65    4942 1051.13  4965.2 1035.11  4983.5 1029.39
    4985 1028.39  5049.1 1029.39    5065 1032.78  5073.9 1037.01  5094.4 1041.73
  5165.2 1047.45  5265.5 1050.57  5385.1 1056.09  5466.1  1064.7  5566.3 1073.52
  5618.1 1078.61  5684.1 1088.26  5753.9 1096.01  5846.1 1101.09  5913.9  1107.1
#Mann= 13 ,-1 , 0
    4492     .07       0    4540     .12       0  4669.5     .07       0
  4863.4     .12       0  4965.2    .033       0  4983.5    .033       0
  5049.1    .033       0    5065     .12       0  5165.2     .12       0
  5265.5    .035       0  5466.1     .12       0  5566.3    .035       0
  5684.1     .07       0
Bank Sta=4983.5,5049.1
XS Rating Curve= 0 ,0
Exp/Cntr=0.3,0.1

Type RM Length L Ch R = 1 ,9081    ,686,686,686
BEGIN DESCRIPTION:
CURRY CREEK 13.0
END DESCRIPTION:
XS GIS Cut Line= 3
        2131325.       13874075.        2130825.       13873875.
      2129799.92     13873877.93
#Sta/Elev= 30
  4467.6 1114.53  4530.9 1100.92  4536.3 1101.66  4553.8 1096.41  4560.5 1092.05
  4565.9 1092.33  4584.7 1086.75  4590.1 1087.72  4614.3 1080.13  4751.7 1063.57
  4805.5 1054.64  4812.2 1053.14  4829.7 1038.52  4866.1 1036.34  4898.4 1030.04
  4939.7 1028.59  4963.9 1026.94  4965.4 1025.94  5029.5 1026.94  5036.1 1030.18
  5056.1 1028.88  5086.1 1040.22  5106.1 1043.67  5205.2 1051.77  5356.1 1057.37
  5586.5 1073.13  5696.1 1083.37  5786.1 1096.12  5906.1 1108.73  6031.2 1114.27
#Mann= 6 ,-1 , 0
  4467.6     .12       0  4939.7     .12       0  4963.9     .05       0
  5029.5     .12       0  5205.2    .035       0  5586.5     .12       0
Bank Sta=4963.9,5029.5
XS Rating Curve= 0 ,0
Exp/Cntr=0.3,0.1

Type RM Length L Ch R = 1 ,8395    ,719,719,719
BEGIN DESCRIPTION:
CURRY CREEK 12.0
END DESCRIPTION:
XS GIS Cut Line= 3
      2131324.97     13873624.98        2130725.       13873225.
      2129924.76     13872445.65
#Sta/Elev= 30
  4278.8 1096.38  4280.6 1096.38  4328.3 1092.48  4384.3 1080.32  4396.7 1079.79
    4459 1068.73  4523.6 1065.66    4756 1046.19    4776 1044.85    4791 1037.91
  4860.9  1029.6  4944.5 1024.01    4946 1023.01  5010.2 1024.01  5042.2 1026.01
  5049.4  1034.3  5056.4 1033.33  5063.5 1039.56  5070.5 1038.26  5077.7 1042.14
  5091.8  1044.1  5162.5 1049.88  5268.5 1053.06  5367.6 1080.22    5410 1101.19
  5445.5 1115.54  5459.6 1127.21  5494.9 1132.46  5770.6 1146.78  6116.9 1151.89
#Mann= 8 ,-1 , 0
  4278.8    .035       0  4280.6     .12       0  4384.3    .035       0
  4396.7     .12       0    4756    .035       0  4860.9     .12       0
  4944.5     .05       0  5010.2     .12       0
Bank Sta=4944.5,5010.2
XS Rating Curve= 0 ,0
Exp/Cntr=0.3,0.1

Type RM Length L Ch R = 1 ,7676    ,713,713,713
BEGIN DESCRIPTION:
CURRY CREEK 11.0
END DESCRIPTION:
XS GIS Cut Line= 3
      2131575.01     13873675.02        2131075.       13872675.
      2130674.97     13872374.97
#Sta/Elev= 30
  3881.2 1112.05  3925.9 1110.26  3992.8  1098.3  3999.2 1097.44  4104.4  1081.7
  4149.3 1076.87  4448.6 1057.27  4622.1 1051.04  4886.3  1037.5  4946.2 1025.85
  4952.4 1017.65  4953.9 1016.65  5018.1 1017.65  5027.4 1021.52  5056.5 1023.36
  5077.4 1035.95  5085.7 1035.84    5092 1042.97  5106.5 1045.44  5112.8 1053.02
  5121.1 1053.67  5127.4  1062.2  5135.7 1062.34    5142 1069.55  5177.4 1092.64
  5221.1 1114.39  5227.4 1126.92    5242 1141.29  5327.4 1149.16  5499.3 1157.28
#Mann= 9 ,-1 , 0
  3881.2     .07       0  3992.8     .12       0  3999.2     .07       0
  4104.4     .12       0  4149.3    .035       0  4622.1     .12       0
  4886.3     .12       0  4952.4     .05       0  5018.1     .12       0
Bank Sta=4952.4,5018.1
XS Rating Curve= 0 ,0
Exp/Cntr=0.3,0.1

Type RM Length L Ch R = 1 ,6963    ,581,581,581
BEGIN DESCRIPTION:
CURRY CREEK 10.0
END DESCRIPTION:
XS GIS Cut Line= 3
      2132124.99     13873474.98        2131725.       13872675.
        2131425.       13872275.
#Sta/Elev= 30
  4109.9 1116.61  4199.3 1110.06  4310.4 1084.29  4335.6 1079.32  4422.1 1066.79
  4543.1 1052.62  4817.2 1040.04  4833.8 1037.59  4847.8 1032.33  4861.8 1034.72
  4878.5 1033.46  4884.1 1034.88  4906.5 1032.07  4923.2 1027.17  4928.8 1027.54
  4945.6 1021.25  4949.1 1016.83  4950.6 1015.83  5014.8 1016.83  5032.4 1019.92
  5040.8 1025.22    5047 1025.08  5061.6 1033.47  5082.4 1034.74  5090.8 1037.66
  5104.3    1046  5111.6 1053.51  5304.3 1080.07  5367.8 1095.82  5504.3 1113.49
#Mann= 7 ,-1 , 0
  4109.9     .12       0  4310.4     .07       0  4335.6     .12       0
  4422.1    .035       0  4817.2     .12       0  4949.1     .05       0
  5014.8     .12       0
Bank Sta=4949.1,5014.8
XS Rating Curve= 0 ,0
Exp/Cntr=0.3,0.1

Type RM Length L Ch R = 1 ,6382    ,781,781,781
BEGIN DESCRIPTION:
CURRY CREEK 9.0
END DESCRIPTION:
XS GIS Cut Line= 3
      2132596.63     13873607.12        2132275.       13872675.
       2131502.5     13872210.59
#Sta/Elev= 30
  4014.3  1132.2  4104.4 1126.23  4158.3 1123.96  4291.6 1112.47  4323.3 1106.74
    4408 1081.69  4434.1 1077.66  4459.7 1071.41  4490.9 1066.81  4598.4 1059.21
  4646.9 1052.68  4709.3 1049.38  4766.4 1043.63    4884 1037.23  4915.7 1034.49
  4937.8 1029.72  4958.8 1024.96  4979.2 1016.48  4990.8 1015.25  4992.3 1014.25
  5056.5 1015.25  5066.4 1024.76  5072.2 1027.33  5124.7 1030.53  5188.8 1041.34
  5394.7 1055.88  5458.8 1062.79  5612.3 1071.39  5700.4  1082.3  5901.7 1101.06
#Mann= 6 ,-1 , 0
  4014.3     .07       0  4104.4     .12       0  4434.1     .07       0
  4937.8     .12       0  4990.8     .05       0  5056.5     .12       0
Bank Sta=4990.8,5056.5
XS Rating Curve= 0 ,0
Exp/Cntr=0.3,0.1

Type RM Length L Ch R = 1 ,5601    ,706,706,706
BEGIN DESCRIPTION:
CURRY CREEK 8.0
END DESCRIPTION:
XS GIS Cut Line= 3
      2133075.05       13872125.        2132575.       13872125.
      2131548.46     13872145.75
#Sta/Elev= 30
  4494.8  1123.1  4644.8    1116  4684.8 1113.35  4704.8 1110.22  4724.8 1104.33
  4764.8 1090.39  4784.8 1081.65  4804.8 1075.46  4844.8 1065.25  4904.8 1053.22
  4914.8 1031.83  4924.8 1027.38  4944.8 1025.16  4974.8 1013.82    4982 1013.01
  4983.5 1012.01  5046.3 1012.01  5047.8 1013.01  5054.9 1023.92  5084.9 1029.61
  5094.9 1034.28  5104.9 1036.36  5124.9 1036.94  5164.9 1043.07  5204.9 1044.58
  5224.9 1046.79    5515 1055.24    5745 1071.14    5835 1075.11  6021.6 1090.89
#Mann= 3 ,-1 , 0
  4494.8     .12       0    4982     .05       0  5047.8     .12       0
Bank Sta=4982,5047.8
XS Rating Curve= 0 ,0
Exp/Cntr=0.3,0.1

Type RM Length L Ch R = 1 ,4895    ,688,688,688
BEGIN DESCRIPTION:
CURRY CREEK 7.0
END DESCRIPTION:
XS GIS Cut Line= 3
        2132825.       13871625.        2132325.       13871525.
      2131273.35     13871702.33
#Sta/Elev= 30
  4495.8 1100.57  4587.6 1093.46  4699.8 1071.69  4842.5 1057.22  4852.7    1038
  4862.9 1028.11  4913.9 1021.42  4954.7 1018.16  4982.9 1009.84  4984.4 1008.84
  5048.7 1009.84    5057 1022.78  5117.3 1034.62  5178.1 1042.79    5239 1045.06
  5335.9 1044.64  5512.3 1048.18  5638.4 1058.88  5754.3  1073.6  5820.7 1079.48
  5867.7 1092.01  5875.3 1095.28  5880.3 1094.93  5908.3  1104.6  5935.8 1111.89
  5940.8 1111.19  5969.1 1118.85  5979.3 1120.78    6030 1123.55  6072.2 1128.35
#Mann= 5 ,-1 , 0
  4495.8     .12       0  4982.9     .05       0  5048.7     .12       0
    5057    .035       0  5820.7     .12       0
Bank Sta=4982.9,5048.7
XS Rating Curve= 0 ,0
Exp/Cntr=0.3,0.1

Type RM Length L Ch R = 1 ,4207    ,692,692,692
BEGIN DESCRIPTION:
CURRY CREEK 6.0
END DESCRIPTION:
XS GIS Cut Line= 3
      2132574.98     13871124.99        2132075.       13870925.
        2131375.       13871025.
#Sta/Elev= 30
  4462.2 1063.59    4522 1060.51  4763.7 1046.29  4800.1 1042.61  4817.6 1039.23
  4824.3 1035.39  4829.7 1036.14  4848.6 1025.07    4854 1027.64  4860.7 1023.12
  4871.5 1020.53  4907.8  1018.7  4914.5 1015.88  4937.4 1014.26  4946.3 1009.83
  4947.8 1008.83  5012.1 1009.83  5041.1 1012.01  5061.3 1020.71    5079 1025.43
    5132 1034.65  5296.6 1037.23  5354.2 1038.74  5379.4 1043.32    5425 1055.52
  5479.4 1063.44  5495.7 1067.45  5566.4 1074.46  5636.8  1100.1  5707.8 1108.26
#Mann= 9 ,-1 , 0
  4462.2    .035       0    4522     .12       0  4946.3     .05       0
  5012.1     .12       0    5079    .035       0  5296.6     .07       0
  5379.4     .12       0  5479.4     .07       0  5636.8     .12       0
Bank Sta=4946.3,5012.1
XS Rating Curve= 0 ,0
Exp/Cntr=0.3,0.1

Type RM Length L Ch R = 1 ,3515    ,732,732,732
BEGIN DESCRIPTION:
CURRY CREEK 5.0
END DESCRIPTION:
XS GIS Cut Line= 3
      2132882.45     13871199.75        2132125.       13870325.
      2131559.03     13869741.52
#Sta/Elev= 30
    3847 1081.51  3969.3 1071.77  4302.7 1050.91  4401.5  1047.8  4501.2 1042.05
  4727.2 1036.33  4925.7 1028.77    4940  1024.5  4947.6 1018.49  4949.7 1004.43
  4951.2 1003.43  5015.7 1004.43  5032.3 1005.55  5053.6 1013.98  5067.8 1015.36
  5096.1 1024.71  5152.7 1035.38    5181  1037.1    5280 1034.29  5294.1 1036.92
  5315.2 1045.49  5371.8  1053.7  5449.7 1061.96  5527.5 1066.04  5612.3 1074.12
  5668.9 1083.74  5711.4 1097.84  5718.3 1101.66  5760.8 1112.01    5817 1117.37
#Mann= 3 ,-1 , 0
    3847    .035       0  4949.7     .05       0  5015.7     .12       0
Bank Sta=4949.7,5015.7
XS Rating Curve= 0 ,0
Exp/Cntr=0.3,0.1

Type RM Length L Ch R = 1 ,2783    ,667,667,667
BEGIN DESCRIPTION:
CURRY CREEK 4.0
END DESCRIPTION:
XS GIS Cut Line= 3
        2132925.     13870925.02        2132825.       13870425.
      2132752.88     13869305.05
#Sta/Elev= 30
  4490.1 1063.38  4668.1 1049.85  4683.9 1049.08  4724.7 1040.42  4755.3  1037.3
  4816.5 1031.35  4836.9 1023.54  4857.3 1025.98  4867.5 1019.49  4875.2  1001.8
  4876.7  1000.8  4941.3  1001.8    4949 1003.89  4969.4 1003.59  4979.6 1005.26
  5050.1 1005.29  5070.2 1015.58  5090.2 1016.95  5100.2 1020.15  5110.3 1025.65
  5130.3  1042.9  5170.4 1059.11  5210.5 1066.23  5234.5 1073.23  5270.6 1088.04
  5320.7 1112.17  5360.8 1120.33  5501.1 1126.37  5698.3 1131.71  6122.3 1134.49
#Mann= 5 ,-1 , 0
  4490.1    .035       0  4668.1     .07       0  4755.3     .12       0
  4875.2     .05       0  4941.3     .12       0
Bank Sta=4875.2,4941.3
XS Rating Curve= 0 ,0
Exp/Cntr=0.3,0.1

Type RM Length L Ch R = 1 ,2116    ,722,722,722
BEGIN DESCRIPTION:
CURRY CREEK 3.0
END DESCRIPTION:
XS GIS Cut Line= 3
        2133225.     13871024.99        2133425.       13870525.
      2133125.01     13869925.03
#Sta/Elev= 30
  4461.9 1075.56  4537.3 1068.36  4833.5 1051.16  4883.3 1046.92  4892.7 1037.16
  4902.1 1031.79  4937.1 1020.03    4956 1008.59  4978.9 1001.65  4985.6  995.24
  4989.7   995.1  4991.2   994.1  5055.8   995.1  5059.1 1002.45  5075.9 1018.08
  5081.5 1015.37  5098.2 1026.32  5120.6 1030.92  5157.4 1031.51  5335.8 1037.67
  5380.8 1044.54  5433.6 1059.24  5506.3 1073.61  5545.5 1086.69    5551 1086.11
  5567.8 1095.51  5573.4 1095.51  5590.2 1106.46  5612.5  1112.2  5671.2 1118.68
#Mann= 6 ,-1 , 0
  4461.9    .035       0  4833.5     .12       0  4989.7     .05       0
  5055.8     .12       0  5157.4    .035       0  5380.8     .12       0
Bank Sta=4989.7,5055.8
XS Rating Curve= 0 ,0
Exp/Cntr=0.3,0.1

Type RM Length L Ch R = 1 ,1394    ,642,642,642
BEGIN DESCRIPTION:
CURRY CREEK 2.0
END DESCRIPTION:
XS GIS Cut Line= 3
      2134574.99     13870724.99        2134075.       13870325.
        2133675.     13869725.01
#Sta/Elev= 30
  4364.6 1105.49  4499.5 1081.33  4556.7 1071.56  4645.2  1064.5  4705.5 1056.89
  4770.4 1048.98  4840.8 1025.66  4848.8 1028.67  4863.2 1026.06  4890.4 1012.05
  4898.4 1011.65  4904.8 1002.49  4912.9  998.51  4958.2  996.25  4959.7  995.25
  5024.3  996.25  5027.4 1013.53    5041 1019.46  5099.5 1033.08  5122.3  1035.5
  5320.4 1039.48  5357.9 1041.36    5373 1047.55  5393.4 1049.05  5489.6 1056.27
  5505.3 1058.29  5574.3 1069.64  5625.4 1081.72  5653.9 1092.89    5726  1105.3
#Mann= 10 ,-1 , 0
  4364.6     .12       0  4499.5     .07       0  4645.2    .035       0
  4705.5     .12       0  4958.2     .05       0  5024.3     .12       0
  5122.3    .035       0  5393.4     .12       0  5489.6    .035       0
  5505.3     .12       0
Bank Sta=4958.2,5024.3
XS Rating Curve= 0 ,0
Exp/Cntr=0.3,0.1

Type RM Length L Ch R = 1 ,752     ,528,528,528
BEGIN DESCRIPTION:
CURRY CREEK 1.0
END DESCRIPTION:
XS GIS Cut Line= 3
      2134924.99     13870574.99        2134625.       13870175.
      2133724.96     13869574.98
#Sta/Elev= 30
  4494.3 1117.72  4550.8  1113.1  4616.2 1100.77  4651.6 1090.77  4692.2 1086.09
  4851.6 1061.65  4866.2 1056.79  4872.4  1051.7  4880.7 1035.94  4903.2 1021.47
  4930.7 1010.07    4937 1009.67  4939.4  995.19  4940.9  994.19  5005.5  995.19
  5030.3 1000.58  5043.9  1008.6  5088.9 1012.59    5116 1025.71  5182.1 1026.15
  5224.1 1039.19  5268.6 1040.81  5276.5 1041.12  5470.5 1041.61  5512.6 1047.83
  5665.8 1055.58    5842 1070.06  5918.2 1081.38  6003.8 1104.26    6076 1112.97
#Mann= 9 ,-1 , 0
  4494.3     .12       0  4550.8     .07       0  4692.2    .035       0
  4903.2     .12       0  4939.4     .05       0  5005.5     .12       0
  5268.6     .07       0  5276.5    .035       0    5842     .12       0
Bank Sta=4939.4,5005.5
XS Rating Curve= 0 ,0
Exp/Cntr=0.3,0.1

Type RM Length L Ch R = 1 ,224     ,0,0,0
BEGIN DESCRIPTION:
CURRY CREEK 0.0
END DESCRIPTION:
XS GIS Cut Line= 3
      2135141.94      13870642.5      2135085.69     13869976.67
      2133743.53     13869359.88
#Sta/Elev= 30
  4331.8 1125.08  4338.5 1124.76  4437.5 1118.69  4474.2 1117.65  4630.4 1091.26
    4801 1072.12  4911.4 1064.73  4931.4 1022.65  4938.4 1018.21  4952.7 1008.29
  5006.6  995.51  5008.1  994.51  5072.7  995.51  5077.8 1001.79  5091.1 1006.55
  5165.8 1020.09  5195.3 1021.79  5274.9 1022.89  5297.9 1026.79  5308.9 1034.16
  5331.9 1040.19  5386.9 1042.45  5636.1 1042.68  5812.5 1050.98  6002.8 1057.05
  6038.1 1061.24  6215.1 1072.82  6282.3 1081.49  6404.5 1105.49  6477.1 1111.64
#Mann= 11 ,-1 , 0
  4331.8    .035       0  4338.5     .12       0  4437.5     .07       0
  4938.4     .12       0  5006.6     .05       0  5072.7     .12       0
  5195.3     .07       0  5386.9    .035       0  5812.5     .12       0
  6038.1    .035       0  6282.3     .12       0
#XS Ineff= 2 , 0
       0                 5181.32       0 1029.13
Permanent Ineff=
       F       F
Bank Sta=5006.6,5072.7
XS Rating Curve= 0 ,0
Exp/Cntr=0.3,0.1

Chan Stop Cuts=-1
Use User Specified Reach Order=0
Composite Channel Slope=5
