--- Cypress Tributary 2.prj (project) ---

Proj Title=Cypress Tributary 2 Base Level Engineering
Current Plan=p01
Default Exp/Contr=0.3,0.1
English Units
Geom File=g01
Flow File=f01
Plan File=p01
BEGIN DESCRIPTION:
Cypress Tributary 2
END DESCRIPTION:

--- Cypress Tributary 2.p01 (plan) ---

Plan Title=Multiple Run
Short Identifier=Multiple
Geom File=g01
Flow File=f01
Subcritical Flow
K Sum by GR= 0
Std Step Tol= 0.01
Critical Tol= 0.01
Num of Std Step Trials= 20
Max Error Tol= 0.3
Flow Tol Ratio= 0.001
Split Flow NTrial= 30
Split Flow Tol= 0.02
Split Flow Ratio= 0.02
Log Output Level= 0
Friction Slope Method= 1
Unsteady Friction Slope Method= 2
Unsteady Bridges Friction Slope Method= 1
Parabolic Critical Depth
Global Vel Dist=  1 , 1 , 1
Global Log Level= 0
CheckData=True
Encroach Param= -1, 0, 0, 0
BEGIN DESCRIPTION:
Multiple Run
END DESCRIPTION:

--- Cypress Tributary 2.f01 (steady flow) ---

Flow Title=Multiple
Number of Profiles=7
Profile Names=10-year,25-year,50-year,1pct_min,100-year,1pct_plu,500-year
River Rch & RM= Cypress Tributar,Reach-1,35520
     412     656     874     567    1131    2257    1869
River Rch & RM= Cypress Tributar,Reach-1,35213
    1186    2014    2804    1891    3773    7527    6755
River Rch & RM= Cypress Tributar,Reach-1,28266
    1729    2985    4198    2854    5695   11364   10380
River Rch & RM= Cypress Tributar,Reach-1,20136
    2230    3891    5512    3770    7522   15009   13879
River Rch & RM= Cypress Tributar,Reach-1,9474
    2992    5318    7627    5277   10530   21010   19893
River Rch & RM= Cypress Tributar,Reach-1,6044
    3293    5871    8435    5845   11662   23268   22095
River Rch & RM= Cypress Tributar,Reach-1,2715
    3371    6008    8630    5978   11927   23798   22582
Boundary for River Rch & Prof#=Cypress Tributar,Reach-1,1
Up Type=0
Dn Type=3
Dn Slope=0.005
Boundary for River Rch & Prof#=Cypress Tributar,Reach-1,2
Up Type=0
Dn Type=3
Dn Slope=0.005
Boundary for River Rch & Prof#=Cypress Tributar,Reach-1,3
Up Type=0
Dn Type=3
Dn Slope=0.005
Boundary for River Rch & Prof#=Cypress Tributar,Reach-1,4
Up Type=0
Dn Type=3
Dn Slope=0.005
Boundary for River Rch & Prof#=Cypress Tributar,Reach-1,5
Up Type=0
Dn Type=3
Dn Slope=0.005
Boundary for River Rch & Prof#=Cypress Tributar,Reach-1,6
Up Type=0
Dn Type=3
Dn Slope=0.005
Boundary for River Rch & Prof#=Cypress Tributar,Reach-1,7
Up Type=0
Dn Type=3
Dn Slope=0.005

--- Cypress Tributary 2.g01 (geometry) ---

Geom Title=Existing Conditions

River Reach=Cypress Tributar,Reach-1
Reach XY= 30
      2149925.00     13898825.00      2150125.00     13895925.00
      2149175.00     13894475.00      2149225.00     13893725.00
      2148925.00     13893475.00      2148325.00     13893525.00
      2148225.19     13893156.72      2148925.11     13891752.32
      2148478.67     13891173.42      2148624.51     13890640.22
      2148376.59     13890331.06      2149024.30     13889685.70
      2148284.01     13888632.02      2148169.48     13887872.57
      2147634.19     13887381.95      2147376.20     13886235.50
      2147771.87     13885773.37      2148480.85     13883472.71
      2149421.25     13882473.45      2149527.24     13881330.93
      2149980.52     13880272.57      2151073.27     13879019.37
      2150674.87     13877502.31      2150874.32     13875938.92
      2150424.28     13875043.27      2151015.43     13874281.55
      2150980.71     13873872.42      2152343.27     13873575.21
      2154361.09     13873624.33      2154925.00     13873325.00

Type RM Length L Ch R = 1,35520,115,115,115
BEGIN DESCRIPTION:
Cypress Tributary 2 67.0
END DESCRIPTION:
XS GIS Cut Line= 3
      2150170.41     13898795.97      2149925.00     13898789.46
      2149704.97     13898800.31
#Sta/Elev= 30
  4754.5 1406.24  4779.9 1404.38  4849.9 1402.03  4880.0 1397.06  4890.0 1395.05
  4900.0 1393.78  4910.0 1393.37  4920.0 1392.21  4940.0 1390.53  4950.0 1390.06
  4970.0 1389.98  4990.0 1389.30  5002.5 1389.25  5008.0 1389.60  5011.0 1388.05
  5011.2 1387.55  5014.7 1387.55  5015.0 1388.05  5040.0 1392.94  5050.1 1395.30
  5060.1 1398.14  5070.1 1400.13  5080.1 1401.57  5100.1 1402.70  5130.2 1402.89
  5150.2 1403.62  5200.2 1403.97  5209.6 1403.71  5214.6 1404.49  5220.3 1404.25
#Mann=3,-1,0
  4754.5    0.12       0  5011.0    0.05       0  5015.0    0.12       0
Bank Sta=5011,5015
Exp/Cntr=0.3,0.1

Type RM Length L Ch R = 1,35405,192,192,192
BEGIN DESCRIPTION:
Cypress Tributary 2 66.0
END DESCRIPTION:
XS GIS Cut Line= 4
      2150102.06     13898730.86      2149968.62     13898674.44
      2149925.00     13898675.00      2149758.51     13898673.37
#Sta/Elev= 30
  4811.5 1403.03  4837.4 1400.98  4842.8 1400.10  4851.7 1397.93  4866.5 1396.65
  4873.5 1395.31  4884.3 1394.71  4890.2 1392.75  4895.7 1392.61  4913.9 1387.70
  4919.4 1388.08  4927.7 1390.40  4937.6 1392.05  4943.1 1390.41  4949.4 1390.73
  4955.6 1390.04  4960.7 1390.04  4970.0 1389.29  4980.0 1387.90  5002.5 1387.66
  5018.0 1386.99  5018.3 1386.49  5021.8 1386.49  5022.0 1386.99  5040.0 1389.90
  5050.0 1392.02  5080.0 1400.37  5100.0 1402.03  5110.0 1402.37  5166.5 1402.62
#Mann=3,-1,0
  4811.5    0.12       0  5018.0    0.05       0  5022.0    0.12       0
Bank Sta=5018,5022
Exp/Cntr=0.3,0.1

Type RM Length L Ch R = 1,35213,170,170,170
BEGIN DESCRIPTION:
Cypress Tributary 2 65.0
END DESCRIPTION:
XS GIS Cut Line= 3
      2150261.60     13898584.39      2149989.86     13898510.14
      2149700.59     13898481.30
#Sta/Elev= 30
  4718.3 1404.44  4745.9 1403.59  4777.5 1403.47  4828.8 1401.79  4846.6 1399.91
  4851.7 1400.18  4870.3 1396.60  4891.4 1394.42  4901.4 1393.91  4926.0 1389.07
  4932.5 1387.41  4942.8 1386.36  4973.9 1384.98  5014.9 1385.55  5023.0 1384.94
  5023.2 1384.44  5026.7 1384.44  5027.0 1384.94  5045.1 1385.13  5065.2 1388.25
  5095.3 1391.64  5101.3 1393.22  5135.5 1394.76  5165.7 1397.44  5195.8 1399.41
  5201.9 1400.54  5207.0 1399.97  5215.9 1400.26  5246.1 1398.65  5290.7 1398.15
#Mann=3,-1,0
  4718.3    0.12       0  5023.0    0.05       0  5027.0    0.12       0
Bank Sta=5023,5027
Exp/Cntr=0.3,0.1

Type RM Length L Ch R = 1,35043,271,271,271
BEGIN DESCRIPTION:
Cypress Tributary 2 64.0
END DESCRIPTION:
XS GIS Cut Line= 3
      2150269.20     13898367.37      2149975.00     13898375.00
      2149729.43     13898404.19
#Sta/Elev= 30
  4705.7 1400.55  4769.9 1400.51  4779.9 1399.93  4806.1 1395.62  4811.1 1395.87
  4839.9 1394.17  4849.9 1391.83  4870.0 1385.30  4880.0 1383.23  4900.0 1381.23
  4910.0 1380.87  4920.0 1382.18  4940.0 1378.88  4961.7 1378.43  4990.0 1375.82
  5008.1 1375.79  5008.3 1375.29  5011.8 1375.29  5012.1 1375.79  5038.8 1376.44
  5060.4 1378.58  5070.5 1381.01  5090.6 1387.44  5110.8 1391.43  5120.8 1391.85
  5126.5 1393.11  5151.1 1395.16  5191.8 1395.75  5214.2 1396.39  5247.3 1395.91
#Mann=5,-1,0
  4705.7    0.12       0  4961.7    0.07       0  5008.1    0.05       0
  5012.1    0.07       0  5191.8    0.12       0
Bank Sta=5008.1,5012.1
Exp/Cntr=0.3,0.1

Type RM Length L Ch R = 1,34772,270,270,270
BEGIN DESCRIPTION:
Cypress Tributary 2 63.0
END DESCRIPTION:
XS GIS Cut Line= 3
      2150293.02     13898156.86      2149925.00     13898125.00
      2149619.06     13898176.24
#Sta/Elev= 30
  4630.6 1394.66  4658.7 1394.43  4698.9 1395.97  4729.0 1394.51  4749.1 1391.97
  4759.1 1387.70  4762.2 1387.12  4769.1 1385.82  4830.2 1380.71  4869.5 1379.54
  4889.6 1379.99  4929.7 1376.22  4938.4 1376.51  4941.4 1375.94  4941.7 1375.44
  4945.4 1375.94  4979.9 1377.28  5000.6 1376.67  5010.1 1378.93  5050.7 1380.72
  5060.8 1381.86  5093.6 1386.97  5101.4 1388.79  5111.5 1389.55  5121.7 1388.85
  5149.2 1388.95  5154.3 1389.59  5172.4 1388.51  5235.1 1388.30  5310.2 1386.71
#Mann=6,-1,0
  4630.6    0.12       0  4762.2   0.035       0  4941.4   0.035       0
  4945.4   0.035       0  5000.6    0.07       0  5235.1    0.12       0
Bank Sta=4941.4,4945.4
Exp/Cntr=0.3,0.1

Type RM Length L Ch R = 1,34502,413,413,413
BEGIN DESCRIPTION:
Cypress Tributary 2 62.0
END DESCRIPTION:
XS GIS Cut Line= 3
      2150255.27     13897924.66      2149875.00     13897875.00
      2149564.30     13897876.05
#Sta/Elev= 30
  4616.5 1390.06  4626.9 1390.27  4647.0 1382.67  4652.3 1382.93  4677.3 1381.49
  4687.4 1381.99  4788.2 1377.94  4852.4 1376.76  4889.1 1376.41  4909.2 1375.00
  4949.6 1374.35  4963.0 1373.62  4989.9 1373.82  4993.1 1373.04  4995.5 1372.46
  4995.7 1371.96  4999.2 1371.96  4999.5 1372.46  5010.0 1372.51  5020.0 1376.80
  5030.0 1377.90  5060.0 1378.86  5090.0 1380.59  5190.0 1380.00  5200.0 1380.49
  5240.0 1379.25  5250.0 1380.18  5271.7 1379.45  5280.0 1378.98  5310.7 1379.53
#Mann=6,-1,0
  4616.5    0.07       0  4852.4   0.035       0  4993.1    0.07       0
  4995.5    0.05       0  4999.5    0.07       0  5271.7    0.12       0
Bank Sta=4995.5,4999.5
Exp/Cntr=0.3,0.1

Type RM Length L Ch R = 1,34089,391,391,391
BEGIN DESCRIPTION:
Cypress Tributary 2 61.0
END DESCRIPTION:
XS GIS Cut Line= 3
      2150359.41     13897577.43      2150025.00     13897525.00
      2149669.20     13897501.10
#Sta/Elev= 30
  4661.5 1373.85  4746.9 1373.72  4827.9 1372.56  4903.5 1369.93  4908.9 1369.38
  4966.1 1368.68  4997.5 1366.30  5002.5 1366.30  5008.0 1365.00  5008.3 1364.50
  5011.8 1364.50  5012.0 1365.00  5020.0 1365.60  5030.1 1368.02  5050.1 1369.56
  5080.2 1368.59  5100.2 1368.69  5140.3 1369.52  5160.4 1370.39  5170.4 1370.24
  5180.4 1372.76  5190.4 1372.64  5200.5 1373.62  5210.5 1373.86  5219.6 1374.88
  5230.5 1374.82  5240.5 1375.64  5260.6 1375.06  5280.6 1375.67  5356.6 1374.71
#Mann=3,-1,0
  4661.5   0.035       0  5008.0   0.035       0  5012.0   0.035       0
Bank Sta=5008,5012
Exp/Cntr=0.3,0.1

Type RM Length L Ch R = 1,33698,391,391,391
BEGIN DESCRIPTION:
Cypress Tributary 2 60.0
END DESCRIPTION:
XS GIS Cut Line= 3
      2150508.75     13897632.98      2150125.00     13897175.00
      2149484.49     13897053.14
#Sta/Elev= 30
  4402.5 1374.78  4411.3 1375.68  4432.1 1375.68  4439.0 1374.48  4460.7 1373.30
  4553.1 1372.22  4559.6 1372.84  4602.5 1371.09  4680.6 1370.87  4758.7 1368.06
  4779.5 1369.18  4865.3 1362.52  4879.6 1362.16  4886.2 1363.08  4893.9 1361.95
  4914.8 1362.15  4929.1 1361.22  4954.0 1361.71  4964.2 1361.47  4990.8 1358.40
  4991.1 1357.90  4994.8 1358.40  5002.5 1358.46  5010.2 1361.04  5025.4 1362.99
  5142.5 1362.68  5207.1 1365.06  5386.8 1365.39  5606.1 1360.60  5652.0 1360.00
#Mann=6,-1,0
  4402.5   0.035       0  4954.0    0.07       0  4990.8    0.05       0
  4994.8    0.07       0  5207.1    0.12       0  5606.1   0.035       0
Bank Sta=4990.8,4994.8
Exp/Cntr=0.3,0.1

Type RM Length L Ch R = 1,33307,392,392,392
BEGIN DESCRIPTION:
Cypress Tributary 2 59.0
END DESCRIPTION:
XS GIS Cut Line= 3
      2150817.80     13896823.97      2150125.00     13896825.00
      2149528.07     13896879.34
#Sta/Elev= 30
  4307.2 1372.81  4445.7 1369.71  4510.0 1367.24  4540.0 1363.47  4560.0 1365.30
  4580.0 1362.56  4620.0 1360.56  4710.0 1360.39  4780.0 1358.08  4850.0 1357.25
  4910.7 1357.59  4960.0 1355.27  4990.0 1352.46  5010.0 1352.97  5028.1 1351.77
  5028.4 1351.27  5032.1 1351.77  5050.2 1355.76  5055.2 1355.04  5060.2 1356.82
  5100.4 1357.53  5150.6 1359.68  5180.7 1359.77  5195.3 1360.69  5240.6 1359.97
  5291.2 1359.91  5331.4 1358.76  5451.9 1361.10  5562.3 1358.60  5599.4 1359.11
#Mann=7,-1,0
  4307.2   0.035       0  4445.7    0.07       0  4910.7    0.12       0
  5028.1    0.05       0  5032.1    0.12       0  5195.3    0.07       0
  5240.6   0.035       0
Bank Sta=5028.1,5032.1
Exp/Cntr=0.3,0.1

Type RM Length L Ch R = 1,32915,321,321,321
BEGIN DESCRIPTION:
Cypress Tributary 2 58.0
END DESCRIPTION:
XS GIS Cut Line= 3
      2150921.95     13896490.63      2150125.00     13896475.00
      2149533.07     13896532.30
#Sta/Elev= 30
  4202.9 1374.35  4209.8 1372.99  4219.9 1369.43  4234.5 1367.77  4259.9 1366.30
  4279.9 1365.70  4289.9 1364.57  4309.9 1365.34  4369.9 1362.86  4425.5 1361.74
  4479.9 1359.59  4539.9 1359.68  4629.9 1356.84  4659.9 1357.49  4669.9 1355.85
  4719.9 1353.32  4810.0 1350.76  4889.9 1349.84  4995.5 1345.22  4995.7 1344.72
  4999.5 1345.22  5020.1 1348.75  5100.5 1352.16  5184.7 1354.28  5190.9 1354.74
  5301.4 1352.40  5383.3 1352.95  5422.0 1353.51  5506.8 1353.00  5594.7 1353.00
#Mann=10,-1,0
  4202.9    0.07       0  4234.5   0.035       0  4259.9    0.07       0
  4425.5   0.035       0  4889.9    0.07       0  4995.5    0.05       0
  4999.5    0.07       0  5184.7   0.035       0  5383.3    0.07       0
  5506.8   0.035       0
Bank Sta=4995.5,4999.5
Exp/Cntr=0.3,0.1

Type RM Length L Ch R = 1,32594,512,512,512
BEGIN DESCRIPTION:
Cypress Tributary 2 57.0
END DESCRIPTION:
XS GIS Cut Line= 3
      2150869.93     13896216.33      2150075.00     13896175.00
      2149470.60     13896289.24
#Sta/Elev= 30
  4204.0 1360.88  4335.8 1357.11  4434.3 1354.92  4489.3 1353.99  4569.4 1354.60
  4579.4 1352.14  4589.4 1351.39  4828.5 1345.68  4974.0 1342.23  4988.0 1341.00
  4988.2 1340.50  4992.0 1341.00  4997.5 1344.19  5002.6 1344.22  5010.2 1346.87
  5031.3 1348.34  5078.5 1347.67  5083.6 1348.25  5101.8 1347.41  5142.5 1348.22
  5227.9 1348.14  5240.7 1347.87  5254.4 1348.69  5285.0 1347.72  5328.8 1347.83
  5429.7 1347.90  5455.3 1348.29  5460.4 1349.19  5468.1 1348.36  5615.1 1347.81
#Mann=11,-1,0
  4204.0   0.035       0  4335.8    0.07       0  4434.3   0.035       0
  4828.5    0.12       0  4974.0    0.07       0  4988.0    0.05       0
  4992.0    0.07       0  5002.6    0.12       0  5227.9    0.07       0
  5328.8   0.035       0  5429.7    0.07       0
Bank Sta=4988,4992
Exp/Cntr=0.3,0.1

Type RM Length L Ch R = 1,32082,665,665,665
BEGIN DESCRIPTION:
Cypress Tributary 2 56.0
END DESCRIPTION:
XS GIS Cut Line= 3
      2150446.29     13895431.59      2150025.00     13895725.00
      2149388.64     13896215.24
#Sta/Elev= 30
  4486.6 1371.76  4527.7 1369.13  4554.5 1366.43  4569.3 1363.27  4590.3 1360.51
  4605.1 1356.82  4640.9 1352.35  4763.1 1343.97  4838.2 1340.15  4928.3 1339.02
  4963.4 1339.37  4986.5 1337.78  5013.6 1337.73  5021.8 1335.58  5028.1 1335.38
  5036.3 1336.11  5042.6 1337.77  5077.9 1337.62  5119.4 1334.38  5119.7 1333.88
  5123.4 1334.38  5135.9 1338.25  5200.2 1341.46  5349.7 1341.45  5505.5 1343.81
  5520.0 1344.79  5604.8 1345.22  5777.3 1346.58  5798.1 1348.18  5803.3 1347.09
#Mann=7,-1,0
  4486.6    0.12       0  4527.7    0.07       0  4838.2   0.035       0
  4928.3    0.12       0  5119.4    0.05       0  5123.4    0.12       0
  5604.8   0.035       0
Bank Sta=5119.4,5123.4
Exp/Cntr=0.3,0.1

Type RM Length L Ch R = 1,31417,413,413,413
BEGIN DESCRIPTION:
Cypress Tributary 2 55.0
END DESCRIPTION:
XS GIS Cut Line= 3
      2150328.23     13895317.02      2149675.00     13895375.00
      2149058.73     13895545.81
#Sta/Elev= 30
  4344.2 1370.45  4367.5 1369.80  4427.8 1364.42  4437.8 1361.55  4487.0 1356.52
  4498.0 1353.78  4508.1 1352.56  4528.2 1351.10  4608.8 1342.61  4628.5 1342.78
  4678.7 1338.46  4749.0 1334.79  4879.5 1333.64  4889.6 1331.26  4896.1 1330.76
  4929.7 1329.09  4979.9 1330.30  5002.6 1329.31  5008.4 1327.80  5008.6 1327.30
  5012.4 1327.80  5017.1 1330.24  5022.3 1330.83  5033.9 1330.34  5083.0 1329.49
  5209.3 1331.31  5277.9 1331.09  5322.6 1332.33  5470.1 1333.78  5639.5 1333.34
#Mann=5,-1,0
  4344.2    0.07       0  4896.1    0.12       0  5008.4    0.05       0
  5012.4    0.12       0  5033.9    0.07       0
Bank Sta=5008.4,5012.4
Exp/Cntr=0.3,0.1

Type RM Length L Ch R = 1,31004,432,432,432
BEGIN DESCRIPTION:
Cypress Tributary 2 54.0
END DESCRIPTION:
XS GIS Cut Line= 3
      2149904.60     13894785.77      2149525.00     13895025.00
      2148922.09     13895480.12
#Sta/Elev= 30
  4551.3 1353.41  4594.5 1351.14  4600.4 1351.82  4673.4 1347.16  4688.6 1345.36
  4709.8 1344.86  4725.1 1343.03  4767.5 1341.96  4782.8 1340.08  4804.0 1339.52
  4834.5 1336.73  4840.5 1333.59  4855.8 1329.71  4861.7 1329.63  4877.0 1324.47
  4896.2 1321.10  4896.4 1320.60  4900.2 1321.10  4919.4 1323.35  4950.9 1323.49
  4977.1 1324.70  4992.4 1321.46  5003.1 1321.14  5013.5 1322.98  5036.4 1323.47
  5050.1 1325.31  5157.1 1325.02  5286.2 1329.05  5506.8 1331.31  5755.4 1332.03
#Mann=4,-1,0
  4551.3    0.12       0  4896.2    0.05       0  4900.2    0.12       0
  4950.9    0.07       0
Bank Sta=4896.2,4900.2
Exp/Cntr=0.3,0.1

Type RM Length L Ch R = 1,30572,379,379,379
BEGIN DESCRIPTION:
Cypress Tributary 2 53.0
END DESCRIPTION:
XS GIS Cut Line= 3
      2149998.34     13894598.27      2149325.00     13894675.00
      2148310.85     13894775.35
#Sta/Elev= 30
  4322.3 1353.26  4454.2 1347.87  4458.4 1347.70  4647.7 1339.29  4708.1 1329.36
  4776.4 1323.11  4819.7 1321.94  4929.5 1318.34  4969.8 1318.83  4989.9 1316.98
  4997.5 1313.91  5002.5 1313.91  5010.0 1314.28  5020.1 1317.28  5060.3 1317.75
  5100.5 1321.65  5213.6 1323.46  5391.6 1322.12  5472.3 1322.24  5555.1 1320.05
  5643.1 1316.62  5713.5 1316.12  5741.6 1313.81  5741.9 1313.31  5745.6 1313.81
  5861.2 1322.03  5866.2 1320.90  5875.6 1322.94  5956.9 1328.85  6019.1 1330.52
#Mann=11,-1,0
  4322.3    0.12       0  4454.2    0.07       0  4458.4    0.12       0
  4819.7    0.07       0  5213.6   0.035       0  5391.6    0.12       0
  5555.1    0.07       0  5741.6    0.05       0  5745.6    0.07       0
  5875.6    0.12       0  5956.9    0.07       0
Bank Sta=5741.6,5745.6
Exp/Cntr=0.3,0.1

Type RM Length L Ch R = 1,30193,425,425,425
BEGIN DESCRIPTION:
Cypress Tributary 2 52.0
END DESCRIPTION:
XS GIS Cut Line= 3
      2149817.75     13894292.72      2149210.15     13894344.80
      2148369.96     13894681.57
#Sta/Elev= 30
  4352.3 1339.47  4375.1 1338.83  4385.2 1337.07  4495.6 1330.47  4525.7 1330.34
  4585.9 1326.78  4736.5 1322.35  4776.6 1320.88  4826.8 1317.49  4878.2 1316.10
  4973.1 1313.99  5008.8 1311.09  5009.0 1310.59  5012.8 1311.09  5021.5 1311.90
  5033.8 1316.19  5043.1 1318.16  5111.8 1320.13  5290.9 1319.50  5375.5 1317.31
  5571.9 1315.60  5689.5 1312.05  5757.5 1315.65  5775.7 1318.85  5781.8 1322.05
  5787.1 1322.09  5797.2 1324.33  5835.6 1327.28  5865.2 1328.10  5867.3 1329.17
#Mann=4,-1,0
  4352.3    0.12       0  4878.2    0.07       0  5008.8    0.05       0
  5012.8    0.07       0
Bank Sta=5008.8,5012.8
Exp/Cntr=0.3,0.1

Type RM Length L Ch R = 1,29768,533,533,533
BEGIN DESCRIPTION:
Cypress Tributary 2 51.0
END DESCRIPTION:
XS GIS Cut Line= 3
      2149762.20     13893976.74      2149175.00     13893975.00
      2148390.72     13894487.16
#Sta/Elev= 30
  4412.8 1335.36  4470.0 1334.59  4490.0 1333.30  4510.0 1330.01  4520.0 1329.28
  4560.0 1328.14  4710.0 1325.50  4823.8 1324.73  4840.0 1324.54  4860.0 1322.31
  4890.0 1316.57  4910.0 1310.79  4920.0 1309.43  4980.0 1309.60  4995.5 1308.04
  4995.7 1307.54  4999.5 1308.04  5007.6 1309.05  5028.6 1309.29  5071.7 1311.80
  5167.2 1311.72  5375.6 1313.82  5621.1 1313.23  5859.9 1309.91  5873.3 1311.05
  5882.4 1314.45  5888.4 1314.81  5895.8 1319.43  5903.5 1322.56  5936.7 1324.80
#Mann=4,-1,0
  4412.8    0.12       0  4823.8    0.07       0  4995.5    0.05       0
  4999.5    0.07       0
Bank Sta=4995.5,4999.5
Exp/Cntr=0.3,0.1

Type RM Length L Ch R = 1,29235,969,969,969
BEGIN DESCRIPTION:
Cypress Tributary 2 50.0
END DESCRIPTION:
XS GIS Cut Line= 3
      2149203.23     13893303.11      2149025.00     13893575.00
      2148296.96     13894438.55
#Sta/Elev= 30
  4674.9 1306.75  4692.0 1306.60  4877.9 1306.82  4941.2 1304.68  4971.4 1305.34
  4990.5 1304.48  4990.7 1303.98  4994.5 1304.48  5035.7 1305.77  5241.2 1305.22
  5354.4 1307.76  5376.4 1308.97  5483.1 1310.61  5489.6 1309.74  5510.4 1310.43
  5567.6 1309.09  5596.2 1309.65  5766.6 1308.21  5795.2 1305.81  5901.8 1310.30
  5908.3 1311.19  5936.9 1311.86  5979.8 1316.04  5986.3 1317.94  6000.6 1318.87
  6007.2 1321.30  6014.9 1321.68  6021.5 1323.55  6064.4 1326.59  6129.5 1328.81
#Mann=4,-1,0
  4674.9    0.12       0  4692.0    0.07       0  4990.5    0.05       0
  4994.5    0.07       0
Bank Sta=4990.5,4994.5
Exp/Cntr=0.3,0.1

Type RM Length L Ch R = 1,28266,331,331,331
BEGIN DESCRIPTION:
Cypress Tributary 2 49.0
END DESCRIPTION:
XS GIS Cut Line= 3
      2149081.71     13893251.04      2148274.60     13893375.17
      2147685.90     13893507.98
#Sta/Elev= 30
  4183.4 1305.01  4211.1 1304.79  4356.1 1304.05  4726.4 1300.46  4938.9 1297.08
  4959.1 1296.31  4970.2 1294.35  4977.2 1291.38  4977.5 1290.88  4981.5 1291.38
  4989.5 1292.41  4997.3 1296.31  5002.4 1296.31  5018.5 1303.68  5030.3 1306.57
  5102.1 1310.10  5115.2 1312.30  5122.6 1314.74  5143.1 1316.01  5158.4 1315.47
  5184.1 1317.01  5250.0 1318.74  5276.4 1321.25  5307.1 1321.75  5358.4 1324.06
  5384.7 1326.80  5419.9 1327.37  5440.4 1328.77  5501.9 1330.55  5603.5 1332.51
#Mann=5,-1,0
  4183.4   0.035       0  4211.1    0.12       0  4356.1    0.07       0
  4977.2    0.05       0  4981.5    0.07       0
Bank Sta=4977.2,4981.5
Exp/Cntr=0.3,0.1

Type RM Length L Ch R = 1,27935,463,463,463
BEGIN DESCRIPTION:
Cypress Tributary 2 48.0
END DESCRIPTION:
XS GIS Cut Line= 3
      2149289.99     13893174.66      2148224.51     13893061.20
      2147703.22     13893007.99
#Sta/Elev= 30
  3928.5 1307.35  3964.6 1306.53  4162.2 1304.10  4261.0 1302.75  4348.2 1302.36
  4458.7 1302.07  4587.2 1301.66  4687.8 1297.69  4746.3 1297.12  4969.3 1294.41
  4979.4 1294.09  4995.1 1291.04  4995.4 1290.54  4999.1 1290.54  4999.4 1291.04
  5002.3 1291.04  5008.2 1294.18  5019.8 1301.96  5029.7 1305.74  5049.8 1309.76
  5079.9 1312.01  5134.8 1313.68  5200.5 1314.71  5270.9 1318.41  5301.1 1321.21
  5338.5 1321.12  5361.4 1322.66  5381.5 1322.18  5431.7 1327.13  5524.0 1328.18
#Mann=12,-1,0
  3928.5    0.12       0  3964.6    0.07       0  4162.2   0.035       0
  4261.0    0.07       0  4348.2    0.12       0  4458.7    0.07       0
  4746.3   0.035       0  4995.1   0.035       0  4999.4   0.035       0
  5019.8    0.07       0  5134.8   0.035       0  5338.5    0.07       0
Bank Sta=4995.1,4999.4
Exp/Cntr=0.3,0.1

Type RM Length L Ch R = 1,27472,566,566,566
BEGIN DESCRIPTION:
Cypress Tributary 2 47.0
END DESCRIPTION:
XS GIS Cut Line= 3
      2149304.21     13893130.81      2148464.24     13892684.68
      2147859.50     13892757.49
#Sta/Elev= 30
  4048.9 1307.25  4103.4 1306.24  4112.3 1306.08  4323.1 1302.45  4392.5 1301.79
  4430.9 1300.63  4436.5 1301.14  4484.6 1300.80  4704.7 1300.57  4779.7 1297.96
  4842.9 1293.86  4872.2 1293.47  4947.1 1292.08  4988.9 1290.00  4989.2 1289.50
  4993.2 1290.00  5039.5 1291.87  5101.6 1292.32  5131.7 1292.31  5190.6 1295.47
  5208.8 1298.75  5213.8 1298.78  5220.8 1300.83  5230.9 1301.76  5271.2 1304.65
  5372.4 1309.35  5412.2 1313.54  5542.3 1318.59  5603.6 1321.47  5609.1 1322.79
#Mann=11,-1,0
  4048.9    0.12       0  4103.4    0.07       0  4112.3   0.035       0
  4323.1    0.12       0  4484.6    0.07       0  4779.7    0.12       0
  4872.2   0.035       0  4988.9   0.035       0  4993.2   0.035       0
  5101.6    0.07       0  5372.4   0.035       0
Bank Sta=4988.9,4993.2
Exp/Cntr=0.3,0.1

Type RM Length L Ch R = 1,26906,428,428,428
BEGIN DESCRIPTION:
Cypress Tributary 2 46.0
END DESCRIPTION:
XS GIS Cut Line= 3
      2149185.27     13892780.09      2148677.49     13892222.84
      2147925.00     13892325.00
#Sta/Elev= 30
  4246.1 1301.26  4334.2 1299.84  4398.7 1298.06  4554.9 1296.85  4674.4 1295.10
  4724.4 1292.79  4823.0 1292.33  4897.1 1290.23  4979.7 1287.22  4998.1 1284.27
  5010.4 1283.35  5010.7 1282.85  5014.8 1283.35  5032.8 1285.83  5055.6 1287.02
  5143.8 1287.38  5164.0 1289.22  5184.2 1286.47  5214.4 1287.88  5258.7 1288.31
  5386.0 1289.97  5486.9 1293.97  5507.1 1296.15  5651.4 1305.38  5708.9 1308.39
  5718.1 1310.09  5723.2 1310.10  5729.1 1312.43  5739.2 1314.46  5759.4 1315.47
#Mann=9,-1,0
  4246.1    0.07       0  4334.2    0.12       0  4554.9    0.07       0
  4897.1    0.12       0  4979.7    0.07       0  5010.4    0.05       0
  5014.8    0.07       0  5258.7   0.035       0  5651.4    0.07       0
Bank Sta=5010.4,5014.8
Exp/Cntr=0.3,0.1

Type RM Length L Ch R = 1,26478,451,451,451
BEGIN DESCRIPTION:
Cypress Tributary 2 45.0
END DESCRIPTION:
XS GIS Cut Line= 3
      2149125.00     13892225.00      2148873.35     13891864.32
      2148074.95     13891925.00
#Sta/Elev= 30
  4560.2 1296.75  4582.5 1297.20  4612.9 1296.35  4653.7 1295.99  4660.1 1295.34
  4682.1 1295.45  4832.8 1291.90  4868.6 1291.89  4922.2 1290.32  4969.8 1288.66
  4984.6 1286.41  4990.7 1283.24  4996.5 1282.05  5006.1 1281.84  5006.5 1281.34
  5010.6 1281.84  5048.5 1283.57  5108.7 1284.73  5210.4 1283.54  5319.3 1285.04
  5379.4 1285.22  5419.6 1284.35  5628.2 1287.00  5660.2 1288.19  5680.3 1287.53
  5730.1 1292.85  5735.1 1292.80  5770.6 1301.39  5787.8 1302.86  5800.7 1303.23
#Mann=8,-1,0
  4560.2    0.07       0  4612.9    0.12       0  4653.7    0.07       0
  4922.2   0.035       0  5006.1   0.035       0  5010.6   0.035       0
  5628.2    0.07       0  5787.8   0.035       0
Bank Sta=5006.1,5010.6
Exp/Cntr=0.3,0.1

Type RM Length L Ch R = 1,26027,1040,1040,1040
BEGIN DESCRIPTION:
Cypress Tributary 2 44.0
END DESCRIPTION:
XS GIS Cut Line= 3
      2149397.60     13891763.92      2148862.39     13891452.00
      2148024.98     13891825.01
#Sta/Elev= 30
  4373.3 1294.98  4397.3 1294.18  4456.0 1294.52  4563.6 1291.54  4746.7 1290.25
  4824.0 1287.88  4859.9 1286.61  4936.1 1284.86  4958.9 1284.04  4974.6 1281.96
  4980.4 1282.63  5000.9 1279.83  5048.8 1280.56  5105.5 1278.74  5105.8 1278.24
  5110.0 1278.74  5131.0 1278.75  5143.2 1280.81  5183.0 1281.19  5197.9 1283.04
  5229.4 1281.89  5501.5 1282.70  5648.5 1284.51  5727.0 1285.39  5750.2 1286.84
  5773.5 1290.30  5825.4 1294.52  5865.7 1302.04  5877.4 1303.21  5909.5 1303.94
#Mann=8,-1,0
  4373.3    0.12       0  4824.0    0.07       0  4859.9    0.12       0
  4936.1    0.07       0  5048.8   0.035       0  5105.5    0.05       0
  5110.0   0.035       0  5648.5    0.07       0
Bank Sta=5105.5,5110
Exp/Cntr=0.3,0.1

Type RM Length L Ch R = 1,24987,495,495,495
BEGIN DESCRIPTION:
Cypress Tributary 2 43.0
END DESCRIPTION:
XS GIS Cut Line= 3
      2149225.00     13891425.00      2148625.24     13890750.08
      2147824.96     13891425.03
#Sta/Elev= 30
  4097.1 1287.93  4407.7 1283.60  4551.1 1279.79  4633.8 1277.62  4694.5 1277.16
  4939.9 1274.64  4982.2 1276.21  4989.8 1275.89  4996.4 1274.02  5003.4 1274.02
  5008.8 1271.87  5009.2 1271.37  5013.4 1271.87  5032.0 1272.09  5039.6 1273.39
  5060.6 1274.28  5067.1 1273.48  5074.8 1275.71  5188.0 1277.43  5216.6 1276.52
  5294.2 1277.42  5329.6 1277.53  5464.7 1278.07  5585.9 1277.84  5855.1 1281.92
  5926.5 1284.50  5968.4 1290.49  5997.6 1293.29  6018.9 1294.94  6046.9 1299.93
#Mann=11,-1,0
  4097.1    0.12       0  4407.7    0.07       0  4551.1   0.035       0
  4633.8    0.07       0  4694.5   0.035       0  5008.8   0.035       0
  5013.4   0.035       0  5294.2   0.035       0  5329.6    0.07       0
  5464.7   0.035       0  5997.6    0.07       0
Bank Sta=5008.8,5013.4
Exp/Cntr=0.3,0.1

Type RM Length L Ch R = 1,24492,1493,1493,1493
BEGIN DESCRIPTION:
Cypress Tributary 2 42.0
END DESCRIPTION:
XS GIS Cut Line= 5
      2149290.75     13891026.22      2148869.80     13890542.51
      2148620.79     13890388.90      2148378.09     13890373.36
      2147619.19     13890488.57
#Sta/Elev= 30
  3823.0 1281.87  3870.4 1282.06  3941.7 1280.73  4089.7 1279.80  4132.5 1280.04
  4140.1 1279.37  4215.9 1278.15  4295.8 1277.32  4338.5 1275.91  4466.6 1275.17
  4516.9 1273.69  4561.1 1274.49  4719.6 1272.01  4822.7 1271.61  4862.8 1272.71
  4912.9 1271.50  4943.0 1272.21  4973.0 1271.19  4980.8 1269.01  4981.1 1268.51
  4985.4 1269.01  4993.1 1269.75  4999.0 1273.22  5013.2 1273.77  5336.9 1271.66
  5417.8 1272.73  5620.1 1273.57  5670.7 1274.89  5708.3 1277.34  5767.6 1276.54
#Mann=4,-1,0
  3823.0    0.12       0  4215.9   0.035       0  4980.8   0.035       0
  4985.4   0.035       0
Bank Sta=4980.8,4985.4
Exp/Cntr=0.3,0.1

Type RM Length L Ch R = 1,22999,485,485,485
BEGIN DESCRIPTION:
Cypress Tributary 2 41.0
END DESCRIPTION:
XS GIS Cut Line= 3
      2149620.28     13889144.72      2148855.08     13889304.97
      2147739.24     13890279.36
#Sta/Elev= 30
  4218.2 1325.20  4315.5 1320.17  4367.2 1311.13  4468.5 1298.43  4611.8 1290.88
  4635.8 1285.73  4662.9 1277.14  4680.6 1274.04  4693.6 1273.45  4714.0 1279.15
  4787.9 1273.09  4846.8 1269.76  4873.9 1265.94  4887.7 1262.44  4959.2 1260.40
  4975.2 1257.70  4986.9 1256.89  4987.4 1256.39  4992.8 1256.89  5007.2 1260.71
  5028.1 1263.40  5064.2 1264.94  5425.7 1266.86  5636.9 1267.59  5645.9 1267.62
  5773.7 1268.89  5797.6 1268.95  5890.5 1269.40  6162.4 1268.43  6481.4 1271.81
#Mann=14,-1,0
  4218.2    0.07       0  4367.2   0.035       0  4468.5    0.07       0
  4787.9    0.12       0  4873.9    0.07       0  4975.2   0.035       0
  4986.9   0.035       0  4992.8   0.035       0  5425.7    0.07       0
  5636.9   0.035       0  5645.9    0.07       0  5773.7   0.035       0
  5797.6    0.07       0  5890.5   0.035       0
Bank Sta=4986.9,4992.8
Exp/Cntr=0.3,0.1

Type RM Length L Ch R = 1,22514,421,421,421
BEGIN DESCRIPTION:
Cypress Tributary 2 40.0
END DESCRIPTION:
XS GIS Cut Line= 4
      2149460.58     13888432.91      2148615.15     13888914.94
      2148571.70     13889103.04      2147620.30     13890068.34
#Sta/Elev= 30
  4026.8 1323.74  4099.5 1321.82  4125.1 1320.85  4142.3 1318.07  4148.3 1315.90
  4214.9 1312.06  4303.7 1307.57  4355.5 1301.56  4445.8 1298.80  4561.3 1295.64
  4654.8 1292.96  4676.7 1290.84  4707.0 1279.61  4728.6 1276.79  4766.1 1268.27
  4839.0 1263.13  4852.5 1264.74  4862.0 1262.35  4942.6 1257.46  4974.2 1253.32
  4974.6 1252.82  4980.1 1253.32  5024.3 1254.89  5067.0 1259.71  5087.5 1260.53
  5270.3 1262.60  5524.4 1263.92  5616.4 1265.63  6210.3 1266.55  6548.4 1269.98
#Mann=11,-1,0
  4026.8    0.07       0  4099.5   0.035       0  4125.1    0.07       0
  4214.9   0.035       0  4445.8    0.07       0  4561.3   0.035       0
  4676.7    0.12       0  4974.2    0.05       0  4980.1    0.12       0
  5087.5    0.07       0  5270.3   0.035       0
Bank Sta=4974.2,4980.1
Exp/Cntr=0.3,0.1

Type RM Length L Ch R = 1,22093,1016,1016,1016
BEGIN DESCRIPTION:
Cypress Tributary 2 39.0
END DESCRIPTION:
XS GIS Cut Line= 3
      2149394.64     13888412.07      2148300.87     13888648.18
      2147385.04     13889831.13
#Sta/Elev= 30
  3878.1 1321.23  3914.6 1315.65  4051.7 1308.49  4082.3 1308.23  4113.0 1305.01
  4177.9 1301.57  4380.9 1294.82  4441.3 1291.52  4471.1 1280.32  4482.4 1277.52
  4501.8 1273.01  4542.7 1268.29  4685.4 1263.26  4864.2 1258.95  4913.5 1253.42
  4951.9 1252.77  4959.8 1251.00  4960.3 1250.50  4965.8 1251.00  4989.8 1252.36
  5115.5 1255.76  5170.1 1257.19  5237.0 1256.69  5305.9 1257.67  5347.5 1260.34
  5525.9 1262.73  5712.4 1263.13  5946.9 1260.69  6210.4 1265.71  6493.1 1268.00
#Mann=10,-1,0
  3878.1   0.035       0  4177.9    0.07       0  4380.9    0.12       0
  4482.4    0.07       0  4685.4    0.12       0  4959.8   0.035       0
  4965.8    0.12       0  4989.8   0.035       0  5115.5    0.07       0
  5237.0    0.12       0
Bank Sta=4959.8,4965.8
Exp/Cntr=0.3,0.1

Type RM Length L Ch R = 1,21077,444,444,444
BEGIN DESCRIPTION:
Cypress Tributary 2 38.0
END DESCRIPTION:
XS GIS Cut Line= 3
      2148453.66     13887693.32      2148054.62     13887755.15
      2147293.91     13888846.13
#Sta/Elev= 30
  4596.2 1261.60  4614.6 1261.60  4834.2 1257.39  4902.3 1252.89  4915.2 1249.67
  4959.1 1247.27  4970.3 1244.13  4979.4 1243.49  5003.0 1247.14  5036.4 1246.34
  5045.8 1243.26  5046.3 1242.76  5051.9 1243.26  5057.6 1245.48  5078.5 1243.74
  5093.4 1247.04  5108.2 1247.76  5207.1 1248.14  5243.6 1250.42  5251.3 1248.71
  5257.4 1250.12  5266.1 1248.80  5301.9 1248.40  5373.4 1250.06  5811.4 1252.18
  5876.9 1251.36  5933.6 1251.86  5991.5 1254.29  6108.9 1257.96  6330.0 1260.71
#Mann=7,-1,0
  4596.2    0.07       0  4614.6    0.12       0  4915.2   0.035       0
  5045.8   0.035       0  5051.9   0.035       0  5991.5    0.07       0
  6108.9    0.12       0
Bank Sta=5045.8,5051.9
Exp/Cntr=0.3,0.1

Type RM Length L Ch R = 1,20633,497,497,497
BEGIN DESCRIPTION:
Cypress Tributary 2 37.0
END DESCRIPTION:
XS GIS Cut Line= 3
      2148324.99     13887475.00      2147755.15     13887454.62
      2147275.00     13888474.99
#Sta/Elev= 30
  4429.8 1258.28  4509.6 1256.07  4608.1 1251.95  4649.9 1246.71  4679.9 1245.81
  4706.7 1246.02  4830.0 1245.30  4860.1 1244.66  4890.1 1242.95  4940.1 1243.33
  4967.1 1240.89  4967.6 1240.39  4973.2 1240.89  4997.6 1242.81  5044.6 1241.75
  5105.7 1242.83  5128.5 1243.92  5225.2 1244.61  5287.8 1246.26  5293.6 1247.12
  5555.4 1248.16  5669.4 1249.50  5715.0 1250.70  5720.5 1251.40  5760.6 1251.37
  5766.1 1252.18  5783.4 1252.27  5796.2 1253.47  5843.1 1254.11  6127.7 1256.55
#Mann=7,-1,0
  4429.8    0.07       0  4509.6   0.035       0  4608.1    0.07       0
  4706.7   0.035       0  4967.1   0.035       0  4973.2   0.035       0
  5843.1    0.07       0
Bank Sta=4967.1,4973.2
Exp/Cntr=0.3,0.1

Type RM Length L Ch R = 1,20136,533,533,533
BEGIN DESCRIPTION:
Cypress Tributary 2 36.0
END DESCRIPTION:
XS GIS Cut Line= 3
      2148324.97     13887274.99      2147500.48     13887089.67
      2146878.62     13887189.63
#Sta/Elev= 30
  4179.7 1257.15  4230.9 1255.60  4295.6 1252.12  4333.4 1249.22  4338.9 1248.10
  4382.2 1245.94  4538.4 1244.55  4630.6 1241.98  4700.7 1240.90  4907.4 1238.88
  4932.5 1238.05  4938.1 1237.08  4958.6 1235.90  4970.2 1234.29  4975.8 1232.87
  4985.9 1232.73  4986.4 1232.23  4992.3 1232.23  4992.8 1232.73  4999.6 1238.27
  5009.9 1239.73  5024.0 1240.84  5060.7 1241.76  5172.1 1241.71  5243.0 1243.35
  5263.3 1243.18  5283.7 1244.00  5374.7 1244.65  5402.4 1245.43  5654.6 1246.18
#Mann=4,-1,0
  4179.7   0.035       0  4970.2    0.07       0  4985.9    0.05       0
  4992.8    0.07       0
Bank Sta=4985.9,4992.8
Exp/Cntr=0.3,0.1

Type RM Length L Ch R = 1,19603,457,457,457
BEGIN DESCRIPTION:
Cypress Tributary 2 35.0
END DESCRIPTION:
XS GIS Cut Line= 4
      2148155.31     13886926.39      2147484.39     13886609.68
      2147142.66     13886551.34      2146734.25     13886551.34
#Sta/Elev= 30
  4197.7 1244.00  4363.9 1241.93  4488.5 1241.62  4520.7 1241.52  4596.0 1239.15
  4640.4 1235.44  4657.4 1235.03  4685.7 1234.90  4702.9 1236.11  4708.4 1235.57
  4927.9 1236.26  4949.1 1235.56  4959.3 1234.39  4976.1 1230.57  4976.6 1230.07
  4983.1 1230.57  4996.0 1232.62  5001.0 1231.82  5021.6 1232.86  5040.4 1233.51
  5050.6 1235.84  5056.1 1239.21  5061.2 1238.08  5081.0 1240.81  5171.3 1243.91
  5493.9 1250.41  5623.9 1250.76  5680.4 1249.72  5692.8 1249.38  5694.7 1249.38
#Mann=8,-1,0
  4197.7   0.035       0  4488.5    0.12       0  4596.0   0.035       0
  4976.1   0.035       0  4983.1   0.035       0  5021.6    0.07       0
  5680.4    0.12       0  5692.8    0.07       0
Bank Sta=4976.1,4983.1
Exp/Cntr=0.3,0.1

Type RM Length L Ch R = 1,19146,500,500,500
BEGIN DESCRIPTION:
Cypress Tributary 2 34.0
END DESCRIPTION:
XS GIS Cut Line= 3
      2147875.00     13886674.99      2147420.78     13886173.25
      2147325.04     13886125.02
#Sta/Elev= 30
  4323.2 1240.64  4351.2 1240.09  4377.5 1238.08  4422.2 1234.47  4464.8 1233.59
  4556.7 1235.02  4592.5 1234.08  4705.4 1234.28  4719.6 1233.76  4790.6 1233.59
  4868.3 1234.01  4875.7 1233.56  4944.6 1233.96  4953.4 1234.04  4974.4 1232.23
  4981.8 1230.28  4988.6 1226.40  4995.4 1225.13  5000.0 1225.13  5000.6 1224.26
  5001.1 1223.76  5007.1 1223.76  5007.6 1224.26  5023.3 1230.57  5026.4 1232.69
  5032.0 1233.60  5040.1 1236.94  5048.7 1241.40  5054.3 1243.08  5107.2 1245.22
#Mann=5,-1,0
  4323.2    0.12       0  4377.5   0.035       0  4944.6    0.07       0
  5000.6    0.05       0  5007.6    0.07       0
Bank Sta=5000.6,5007.6
Exp/Cntr=0.3,0.1

Type RM Length L Ch R = 1,18646,461,461,461
BEGIN DESCRIPTION:
Cypress Tributary 2 33.0
END DESCRIPTION:
XS GIS Cut Line= 3
      2148424.98     13886524.98      2147745.60     13885805.16
      2147425.01     13885775.00
#Sta/Elev= 30
  4010.2 1245.22  4017.3 1244.41  4021.2 1244.69  4059.7 1243.60  4066.6 1243.99
  4109.1 1240.45  4154.9 1237.64  4201.3 1236.17  4328.4 1234.53  4378.1 1232.59
  4413.3 1232.30  4477.2 1229.16  4547.6 1230.65  4611.6 1230.31  4781.1 1231.10
  4972.4 1229.25  4986.5 1227.75  5002.8 1228.26  5007.1 1227.66  5007.6 1227.16
  5014.1 1227.66  5055.5 1227.85  5101.0 1229.73  5140.2 1229.63  5181.4 1230.69
  5201.5 1232.27  5221.6 1234.85  5251.7 1240.55  5267.7 1242.81  5322.0 1244.47
#Mann=6,-1,0
  4010.2   0.035       0  4021.2    0.07       0  4154.9   0.035       0
  5007.1   0.035       0  5014.1   0.035       0  5140.2    0.07       0
Bank Sta=5007.1,5014.1
Exp/Cntr=0.3,0.1

Type RM Length L Ch R = 1,18185,500,500,500
BEGIN DESCRIPTION:
Cypress Tributary 2 32.0
END DESCRIPTION:
XS GIS Cut Line= 3
      2148524.98     13886524.97      2147824.84     13885402.07
      2147525.02     13885425.00
#Sta/Elev= 30
  3676.7 1245.16  3748.0 1244.33  3836.6 1238.08  3909.6 1236.13  4061.2 1234.67
  4162.2 1231.54  4220.0 1231.70  4250.7 1229.84  4308.5 1228.44  4371.1 1228.17
  4512.6 1227.12  4678.4 1228.41  4786.3 1227.97  4859.5 1224.30  4880.7 1226.88
  4890.2 1225.00  4896.1 1226.49  4917.3 1227.48  4969.2 1226.72  4990.4 1224.32
  4991.8 1223.10  4992.3 1222.60  4998.9 1223.10  5104.6 1228.37  5150.3 1232.90
  5250.6 1233.35  5260.6 1241.28  5270.6 1243.40  5286.1 1243.62  5300.7 1243.63
#Mann=8,-1,0
  3676.7   0.035       0  3836.6    0.07       0  3909.6   0.035       0
  4061.2    0.07       0  4371.1   0.035       0  4991.8   0.035       0
  4998.9   0.035       0  5286.1    0.07       0
Bank Sta=4991.8,4998.9
Exp/Cntr=0.3,0.1

Type RM Length L Ch R = 1,17685,499,499,499
BEGIN DESCRIPTION:
Cypress Tributary 2 31.0
END DESCRIPTION:
XS GIS Cut Line= 3
      2148975.03     13885575.02      2147978.76     13884976.56
      2147625.04     13885124.98
#Sta/Elev= 30
  3837.8 1237.14  3888.4 1235.40  3931.2 1231.02  3993.0 1228.89  4036.0 1228.47
  4156.0 1222.77  4348.9 1216.36  4385.8 1216.99  4394.2 1215.78  4394.7 1215.28
  4401.3 1215.78  4421.1 1218.07  4486.8 1220.50  4531.7 1220.10  4603.4 1222.05
  4654.4 1220.29  4689.4 1222.13  4879.3 1221.64  4910.4 1223.74  4931.8 1221.39
  4949.3 1221.08  4974.6 1218.38  5014.9 1220.45  5056.7 1221.00  5165.0 1223.94
  5210.1 1224.89  5284.2 1228.50  5321.5 1230.06  5351.1 1232.99  5383.6 1233.31
#Mann=10,-1,0
  3837.8    0.07       0  3993.0   0.035       0  4156.0    0.12       0
  4394.2    0.05       0  4401.3    0.12       0  4531.7   0.035       0
  4949.3    0.07       0  5056.7    0.12       0  5165.0    0.07       0
  5284.2   0.035       0
Bank Sta=4394.2,4401.3
Exp/Cntr=0.3,0.1

Type RM Length L Ch R = 1,17186,468,468,468
BEGIN DESCRIPTION:
Cypress Tributary 2 30.0
END DESCRIPTION:
XS GIS Cut Line= 3
      2148824.98     13885324.98      2148024.56     13884520.27
      2147725.02     13884575.00
#Sta/Elev= 30
  3865.0 1224.96  3894.6 1223.48  4062.9 1217.76  4084.2 1215.20  4119.5 1213.83
  4303.4 1219.08  4423.6 1217.12  4473.1 1218.71  4572.6 1218.63  4592.0 1218.64
  4708.1 1218.48  4735.1 1218.52  4777.2 1219.54  4798.3 1217.80  4833.7 1217.91
  4843.7 1216.53  4865.9 1217.09  4961.0 1213.66  4975.1 1212.40  4982.2 1210.08
  4989.3 1209.83  4992.6 1207.30  4993.1 1206.80  4999.7 1207.30  5009.7 1207.92
  5025.5 1212.11  5070.7 1215.38  5213.0 1217.69  5272.8 1221.94  5304.5 1222.94
#Mann=11,-1,0
  3865.0    0.07       0  3894.6    0.12       0  4572.6   0.035       0
  4592.0    0.12       0  4708.1   0.035       0  4735.1    0.07       0
  4843.7   0.035       0  4865.9    0.07       0  4992.6    0.05       0
  4999.7    0.07       0  5025.5    0.12       0
Bank Sta=4992.6,4999.7
Exp/Cntr=0.3,0.1

Type RM Length L Ch R = 1,16718,497,497,497
BEGIN DESCRIPTION:
Cypress Tributary 2 29.0
END DESCRIPTION:
XS GIS Cut Line= 4
      2148996.04     13885184.90      2148500.98     13884484.93
      2148273.57     13884171.11      2147821.89     13883939.94
#Sta/Elev= 30
  3755.1 1226.84  3829.5 1223.51  3904.1 1218.57  4000.7 1215.03  4114.1 1210.13
  4221.2 1211.67  4244.6 1207.61  4286.4 1211.15  4328.1 1209.86  4385.6 1211.42
  4458.8 1214.35  4560.4 1213.64  4595.4 1211.36  4720.5 1211.87  4816.4 1210.54
  4982.9 1203.03  4989.0 1200.23  4994.5 1194.50  5000.0 1194.50  5003.2 1189.39
  5006.0 1186.89  5006.5 1186.39  5013.2 1186.89  5032.1 1194.97  5042.0 1201.52
  5054.6 1204.75  5086.4 1207.38  5156.7 1208.20  5301.7 1207.61  5507.4 1214.68
#Mann=12,-1,0
  3755.1    0.07       0  3829.5   0.035       0  3904.1    0.12       0
  4000.7    0.07       0  4328.1    0.12       0  4385.6    0.07       0
  4560.4    0.12       0  4720.5   0.035       0  4816.4    0.07       0
  5006.0    0.05       0  5013.2    0.07       0  5156.7    0.12       0
Bank Sta=5006,5013.2
Exp/Cntr=0.3,0.1

Type RM Length L Ch R = 1,16221,440,440,440
BEGIN DESCRIPTION:
Cypress Tributary 2 28.0
END DESCRIPTION:
XS GIS Cut Line= 3
      2148475.00     13883775.00      2148374.55     13883711.18
      2148274.98     13883624.98
#Sta/Elev= 30
  4881.0 1201.65  4888.6 1201.24  4894.5 1201.43  4903.9 1200.25  4909.8 1200.15
  4925.0 1194.08  4931.0 1193.88  4940.2 1189.62  4946.2 1186.08  4961.5 1185.36
  4988.6 1185.31  4996.8 1184.24  5000.2 1184.24  5000.7 1183.74  5007.1 1183.74
  5007.6 1184.24  5018.2 1184.65  5025.8 1187.42  5032.4 1188.26  5039.1 1191.07
  5046.7 1193.54  5053.3 1193.81  5060.9 1195.70  5075.2 1197.56  5081.8 1198.05
  5089.4 1199.47  5117.9 1201.34  5124.5 1201.92  5128.4 1202.67  5131.7 1202.67
#Mann=3,-1,0
  4881.0    0.12       0  5000.2    0.05       0  5007.6    0.12       0
Bank Sta=5000.2,5007.6
Exp/Cntr=0.3,0.1

Type RM Length L Ch R = 1,15781,498,498,498
BEGIN DESCRIPTION:
Cypress Tributary 2 27.0
END DESCRIPTION:
XS GIS Cut Line= 3
      2148775.02     13883475.01      2148576.03     13883339.06
      2148475.00     13883325.00
#Sta/Elev= 30
  4759.0 1195.17  4766.5 1195.05  4787.5 1193.97  4802.4 1192.77  4808.4 1191.73
  4817.3 1190.97  4838.3 1187.45  4844.3 1185.58  4853.2 1184.37  4859.2 1182.84
  4880.2 1181.57  4925.0 1181.18  4945.9 1179.80  4952.8 1179.62  4966.9 1177.66
  4975.8 1177.08  4981.8 1175.62  4985.4 1175.29  4985.9 1174.79  4992.3 1174.79
  4992.8 1175.29  4996.8 1177.48  4999.2 1179.51  5003.0 1179.51  5031.3 1188.83
  5051.5 1192.35  5071.7 1195.12  5081.8 1195.50  5091.9 1196.52  5102.0 1196.82
#Mann=3,-1,0
  4759.0   0.035       0  4985.4   0.035       0  4992.8   0.035       0
Bank Sta=4985.4,4992.8
Exp/Cntr=0.3,0.1

Type RM Length L Ch R = 1,15283,481,481,481
BEGIN DESCRIPTION:
Cypress Tributary 2 26.0
END DESCRIPTION:
XS GIS Cut Line= 3
      2149024.98     13883124.97      2148955.07     13883045.02
      2148674.99     13882975.00
#Sta/Elev= 30
  4893.8 1185.68  4897.1 1185.68  4900.9 1184.68  4907.5 1184.33  4915.1 1183.26
  4921.8 1182.98  4929.4 1181.40  4936.0 1181.11  4950.2 1179.31  4964.5 1175.43
  4978.7 1173.82  4992.9 1168.81  4993.4 1168.31  4999.9 1168.31  5000.4 1168.81
  5010.4 1169.35  5018.1 1170.80  5023.3 1172.31  5041.3 1174.61  5069.6 1175.89
  5082.5 1176.74  5100.6 1176.88  5113.5 1178.00  5134.1 1177.65  5154.7 1178.24
  5195.9 1181.64  5224.3 1186.42  5237.2 1187.94  5270.7 1189.94  5288.7 1191.48
#Mann=4,-1,0
  4893.8    0.07       0  4992.9    0.05       0  5000.4    0.07       0
  5069.6    0.12       0
Bank Sta=4992.9,5000.4
Exp/Cntr=0.3,0.1

Type RM Length L Ch R = 1,14802,497,497,497
BEGIN DESCRIPTION:
Cypress Tributary 2 25.0
END DESCRIPTION:
XS GIS Cut Line= 3
      2149624.99     13882775.00      2149274.13     13882709.64
      2148925.04     13882675.00
#Sta/Elev= 30
  4643.1 1187.47  4674.5 1186.34  4795.7 1174.87  4816.0 1170.72  4832.7 1164.96
  4866.9 1164.82  4890.6 1166.07  4907.6 1170.85  4927.9 1172.09  4968.6 1171.35
  4978.8 1169.79  4988.9 1164.74  4991.4 1164.93  4996.0 1165.27  5015.5 1164.14
  5016.0 1163.64  5023.0 1164.14  5029.3 1167.62  5039.3 1170.00  5049.4 1171.21
  5079.5 1171.88  5089.6 1173.21  5101.1 1172.13  5136.3 1171.78  5180.0 1171.41
  5202.0 1170.46  5210.2 1170.86  5260.4 1177.67  5297.9 1180.78  5350.8 1182.69
#Mann=5,-1,0
  4643.1    0.12       0  4991.4    0.07       0  5015.5    0.05       0
  5023.0    0.07       0  5136.3    0.12       0
Bank Sta=5015.5,5023
Exp/Cntr=0.3,0.1

Type RM Length L Ch R = 1,14305,460,460,460
BEGIN DESCRIPTION:
Cypress Tributary 2 24.0
END DESCRIPTION:
XS GIS Cut Line= 3
      2149891.17     13882554.45      2149424.55     13882264.81
      2148672.40     13882245.41
#Sta/Elev= 30
  4450.8 1189.91  4471.2 1189.04  4566.1 1185.86  4585.1 1185.51  4665.9 1183.33
  4687.2 1179.89  4708.4 1177.76  4802.9 1172.87  4870.0 1170.44  4891.5 1168.22
  4912.8 1164.18  4964.2 1161.00  4970.6 1159.53  4976.5 1159.58  4991.9 1157.71
  4992.5 1157.05  4993.0 1156.55  5001.1 1157.05  5029.6 1163.73  5049.6 1165.35
  5149.6 1166.44  5219.6 1170.51  5349.7 1173.06  5379.7 1172.97  5529.7 1176.59
  5574.5 1179.86  5579.7 1181.03  5619.8 1184.75  5719.8 1190.31  5752.4 1190.83
#Mann=6,-1,0
  4450.8    0.07       0  4471.2    0.12       0  4566.1    0.07       0
  4585.1    0.12       0  4992.5    0.05       0  5001.1    0.12       0
Bank Sta=4992.5,5001.1
Exp/Cntr=0.3,0.1

Type RM Length L Ch R = 1,13845,241,241,241
BEGIN DESCRIPTION:
Cypress Tributary 2 23.0
END DESCRIPTION:
XS GIS Cut Line= 3
      2149925.00     13882175.00      2149514.19     13881834.63
      2148675.86     13881880.82
#Sta/Elev= 30
  4466.5 1182.61  4469.3 1182.61  4494.5 1181.42  4537.5 1175.87  4558.9 1174.56
  4641.9 1169.60  4757.6 1166.58  4891.6 1165.13  4897.9 1165.22  4963.4 1163.72
  4992.0 1160.57  4996.2 1157.48  5002.1 1157.48  5004.9 1155.86  5005.4 1155.36
  5013.1 1155.36  5013.6 1155.86  5039.2 1158.38  5069.3 1158.51  5109.4 1160.99
  5139.4 1165.30  5210.7 1167.89  5282.0 1170.51  5309.6 1170.61  5530.0 1173.60
  5630.1 1176.21  5710.3 1180.35  5730.3 1182.72  5800.4 1184.74  5839.6 1187.34
#Mann=10,-1,0
  4466.5    0.07       0  4469.3   0.035       0  4558.9    0.07       0
  4641.9   0.035       0  4891.6    0.07       0  4897.9    0.12       0
  5004.9    0.05       0  5013.6    0.12       0  5210.7    0.07       0
  5309.6    0.12       0
Bank Sta=5004.9,5013.6
Exp/Cntr=0.3,0.1

Type RM Length L Ch R = 1,13604,542,542,542
BEGIN DESCRIPTION:
Cypress Tributary 2 22.0
END DESCRIPTION:
XS GIS Cut Line= 3
      2150247.40     13881679.61      2149297.22     13881596.26
      2148642.97     13881608.76
#Sta/Elev= 30
  4223.9 1172.22  4398.3 1173.59  4417.0 1172.99  4467.2 1169.42  4487.3 1165.46
  4537.5 1162.74  4735.0 1162.03  4828.6 1161.20  4858.7 1162.04  4879.3 1160.72
  4898.9 1159.53  4929.0 1155.89  4949.1 1156.23  4959.1 1155.31  4974.8 1155.04
  4975.3 1154.54  4983.0 1154.54  4983.5 1155.04  4999.3 1157.47  5017.4 1164.17
  5079.6 1165.74  5210.0 1167.82  5230.0 1167.50  5251.4 1168.26  5448.8 1171.62
  5540.0 1172.88  5640.0 1176.17  5710.0 1180.93  5740.1 1184.52  5832.1 1188.62
#Mann=8,-1,0
  4223.9    0.07       0  4398.3    0.12       0  4735.0    0.07       0
  4879.3    0.12       0  4974.8    0.05       0  4983.5    0.12       0
  5251.4    0.07       0  5448.8    0.12       0
Bank Sta=4974.8,4983.5
Exp/Cntr=0.3,0.1

Type RM Length L Ch R = 1,13062,595,595,595
BEGIN DESCRIPTION:
Cypress Tributary 2 21.0
END DESCRIPTION:
XS GIS Cut Line= 4
      2150150.00     13881600.00      2149633.43     13881119.06
      2149332.47     13881192.48      2148565.22     13881421.57
#Sta/Elev= 30
  4294.2 1172.03  4331.6 1170.99  4386.0 1169.55  4407.6 1167.73  4421.7 1164.99
  4442.7 1164.42  4492.3 1161.12  4519.4 1160.47  4753.8 1159.46  4816.5 1158.78
  4853.1 1159.18  4959.1 1153.46  4973.3 1153.64  4994.8 1151.63  4994.9 1151.07
  4995.4 1150.57  5003.7 1151.07  5019.0 1152.57  5045.4 1159.13  5060.1 1159.70
  5128.8 1161.40  5566.1 1166.35  5648.1 1167.03  5734.2 1168.59  5857.7 1173.51
  5881.1 1175.55  5962.3 1178.98  6000.7 1179.67  6033.8 1182.32  6110.5 1185.48
#Mann=10,-1,0
  4294.2    0.07       0  4331.6    0.12       0  4519.4   0.035       0
  4753.8    0.07       0  4816.5    0.12       0  4994.9    0.05       0
  5003.7    0.12       0  5566.1   0.035       0  5648.1    0.07       0
  5734.2    0.12       0
Bank Sta=4994.9,5003.7
Exp/Cntr=0.3,0.1

Type RM Length L Ch R = 1,12467,710,710,710
BEGIN DESCRIPTION:
Cypress Tributary 2 20.0
END DESCRIPTION:
XS GIS Cut Line= 4
      2150233.46     13881314.18      2149874.64     13880606.67
      2149299.28     13880838.68      2148588.33     13881254.29
#Sta/Elev= 30
  4206.7 1162.37  4346.5 1159.04  4391.0 1158.05  4719.4 1156.83  4854.6 1157.68
  4919.8 1156.50  4942.1 1153.70  4947.7 1149.93  4975.0 1147.56  4975.5 1147.06
  4983.8 1147.56  5007.0 1149.79  5012.3 1149.02  5021.2 1150.22  5066.0 1152.49
  5084.8 1154.27  5090.2 1153.99  5096.7 1154.98  5138.5 1156.62  5466.1 1160.13
  5648.6 1159.92  5811.3 1161.63  5927.5 1162.18  6133.7 1164.53  6227.7 1166.56
  6250.8 1167.50  6278.3 1169.97  6321.3 1172.36  6389.8 1174.22  6443.9 1176.57
#Mann=7,-1,0
  4206.7    0.12       0  4346.5   0.035       0  4854.6    0.12       0
  4975.0    0.05       0  4983.8    0.12       0  5811.3    0.07       0
  5927.5    0.12       0
Bank Sta=4975,4983.8
Exp/Cntr=0.3,0.1

Type RM Length L Ch R = 1,11757,634,634,634
BEGIN DESCRIPTION:
Cypress Tributary 2 19.0
END DESCRIPTION:
XS GIS Cut Line= 4
      2150250.00     13880800.03      2150189.33     13880009.53
      2149853.83     13880067.38      2149006.23     13880648.92
#Sta/Elev= 30
  4208.1 1155.86  4524.1 1154.35  4814.9 1151.60  4875.1 1150.39  4895.1 1150.83
  4935.3 1150.20  4975.4 1147.47  4991.9 1145.39  4992.4 1144.89  5000.7 1145.39
  5015.5 1145.51  5035.8 1147.29  5056.1 1150.06  5061.9 1151.87  5066.9 1149.77
  5076.4 1151.90  5086.5 1152.33  5096.7 1150.95  5127.0 1151.15  5198.1 1152.03
  5375.8 1150.82  5698.6 1153.46  5806.2 1155.11  5842.1 1154.90  5934.8 1156.52
  6079.7 1155.63  6199.6 1156.44  6245.5 1156.04  6321.7 1156.82  6369.3 1156.93
#Mann=6,-1,0
  4208.1   0.035       0  4991.9   0.035       0  5000.7   0.035       0
  5127.0    0.12       0  6199.6    0.07       0  6321.7   0.035       0
Bank Sta=4991.9,5000.7
Exp/Cntr=0.3,0.1
