--- Guadalupe Tributary 36.prj (project) ---

Proj Title=Guadalupe Tributary 36 Base Level Engineering
Current Plan=p01
Default Exp/Contr=0.3,0.1
English Units
Geom File=g01
Flow File=f01
Plan File=p01
BEGIN DESCRIPTION:
Guadalupe Tributary 36
END DESCRIPTION:

--- Guadalupe Tributary 36.p01 (plan) ---

Plan Title=Multiple Run
Short Identifier=Multiple
Geom File=g01
Flow File=f01
Subcritical Flow
K Sum by GR= 0
Std Step Tol= 0.01
Critical Tol= 0.01
Num of Std Step Trials= 20
Max Error Tol= 0.3
Flow Tol Ratio= 0.001
Split Flow NTrial= 30
Split Flow Tol= 0.02
Split Flow Ratio= 0.02
Log Output Level= 0
Friction Slope Method= 1
Unsteady Friction Slope Method= 2
Unsteady Bridges Friction Slope Method= 1
Parabolic Critical Depth
Global Vel Dist=  1 , 1 , 1
Global Log Level= 0
CheckData=True
Encroach Param= -1, 0, 0, 0
BEGIN DESCRIPTION:
Multiple Run
END DESCRIPTION:

--- Guadalupe Tributary 36.f01 (steady flow) ---

Flow Title=Multiple
Number of Profiles=7
Profile Names=10-year,25-year,50-year,1pct_min,100-year,1pct_plu,500-year
River Rch & RM= Guadalupe Tribut,Reach-1,30155
    2035    3575    5092    3510    7003   13973   13108
River Rch & RM= Guadalupe Tribut,Reach-1,23531
    2495    4441    6381    4433    8844   17646   16825
River Rch & RM= Guadalupe Tribut,Reach-1,21664
    3046    5441    7835    5451   10876   21700   20746
River Rch & RM= Guadalupe Tribut,Reach-1,17211
    3554    6387    9233    6444   12858   25655   24692
River Rch & RM= Guadalupe Tribut,Reach-1,14936
    3799    6829    9873    6889   13744   27424   26379
River Rch & RM= Guadalupe Tribut,Reach-1,11793
    3970    7109   10250    7128   14222   28376   27113
Boundary for River Rch & Prof#=Guadalupe Tribut,Reach-1,1
Up Type=0
Dn Type=3
Dn Slope=0.005
Boundary for River Rch & Prof#=Guadalupe Tribut,Reach-1,2
Up Type=0
Dn Type=3
Dn Slope=0.005
Boundary for River Rch & Prof#=Guadalupe Tribut,Reach-1,3
Up Type=0
Dn Type=3
Dn Slope=0.005
Boundary for River Rch & Prof#=Guadalupe Tribut,Reach-1,4
Up Type=0
Dn Type=3
Dn Slope=0.005
Boundary for River Rch & Prof#=Guadalupe Tribut,Reach-1,5
Up Type=0
Dn Type=3
Dn Slope=0.005
Boundary for River Rch & Prof#=Guadalupe Tribut,Reach-1,6
Up Type=0
Dn Type=3
Dn Slope=0.005
Boundary for River Rch & Prof#=Guadalupe Tribut,Reach-1,7
Up Type=0
Dn Type=3
Dn Slope=0.005

--- Guadalupe Tributary 36.g01 (geometry) ---

Geom Title=Existing Conditions

River Reach=Guadalupe Tribut,Reach-1
Reach XY= 30
      2198325.00     13852525.00      2198772.69     13853219.18
      2200584.79     13853785.52      2201244.54     13854795.51
      2202372.70     13855669.17      2204101.87     13855701.18
      2204921.26     13856676.56      2204880.83     13857877.30
      2205772.65     13858980.52      2205644.41     13860195.13
      2206774.90     13860367.21      2207515.13     13860025.88
      2208122.84     13860580.45      2207972.42     13861370.05
      2208321.83     13860932.51      2209263.77     13861064.98
      2209269.91     13861527.30      2208638.27     13862061.31
      2208765.89     13862281.73      2208426.67     13862580.67
      2208664.77     13862864.65      2211305.02     13862874.96
      2211675.00     13863067.92      2212209.84     13862875.38
      2212969.92     13863325.86      2213823.98     13862878.45
      2213968.12     13863375.04      2213576.69     13863430.63
      2213582.08     13864525.03      2214025.00     13865025.00

Type RM Length L Ch R = 1,30155,417,417,417
BEGIN DESCRIPTION:
Guadalupe Tributary 36 47.0
END DESCRIPTION:
XS GIS Cut Line= 3
      2198275.03     13852824.97      2198425.00     13852675.00
      2198824.99     13852475.00
#Sta/Elev= 30
  4792.9 1069.38  4835.3 1066.72  4863.6 1061.78  4891.9 1055.43  4906.0 1053.13
  4934.3 1050.75  4974.3 1048.72  4984.6 1047.88  4990.9 1047.34  4999.4 1044.91
  4999.7 1044.41  5003.3 1044.41  5003.5 1044.91  5007.8 1044.91  5049.7 1049.61
  5060.8 1049.55  5139.2 1052.34  5175.5 1052.71  5183.9 1053.42  5228.6 1054.42
  5287.3 1058.75  5304.1 1061.79  5309.7 1061.90  5326.4 1065.87  5354.4 1070.42
  5376.7 1075.81  5393.5 1081.65  5399.1 1081.85  5409.3 1083.60  5452.2 1089.49
#Mann=7,-1,0
  4792.9    0.07       0  4974.3   0.035       0  4984.6    0.07       0
  4999.4    0.05       0  5003.5    0.07       0  5060.8    0.12       0
  5409.3    0.07       0
Bank Sta=4999.4,5003.5
Exp/Cntr=0.3,0.1

Type RM Length L Ch R = 1,29738,420,420,420
BEGIN DESCRIPTION:
Guadalupe Tributary 36 46.0
END DESCRIPTION:
XS GIS Cut Line= 3
      2198525.01     13853075.00      2198625.00     13853025.00
      2198975.02     13852674.98
#Sta/Elev= 30
  4888.0 1067.56  4890.8 1067.56  4910.4 1064.07  4918.7 1061.22  4924.3 1060.55
  4932.7 1055.37  4941.1 1048.85  4955.1 1042.91  4989.4 1039.30  4989.6 1038.80
  4993.2 1038.80  4993.5 1039.30  4997.0 1041.40  5003.3 1041.40  5070.5 1046.11
  5084.6 1046.87  5105.9 1046.97  5195.5 1050.62  5240.2 1052.43  5268.5 1054.10
  5296.8 1056.52  5310.9 1058.78  5318.0 1060.96  5325.1 1061.82  5353.3 1068.28
  5367.5 1070.86  5381.6 1074.33  5409.9 1082.36  5452.3 1089.33  5494.8 1093.07
#Mann=4,-1,0
  4888.0   0.035       0  4989.4   0.035       0  4993.5   0.035       0
  5195.5    0.12       0
Bank Sta=4989.4,4993.5
Exp/Cntr=0.3,0.1

Type RM Length L Ch R = 1,29318,501,501,501
BEGIN DESCRIPTION:
Guadalupe Tributary 36 45.0
END DESCRIPTION:
XS GIS Cut Line= 3
      2198824.98     13853375.02      2198925.00     13853275.00
      2199175.02     13852874.96
#Sta/Elev= 30
  4859.1 1064.28  4862.7 1064.28  4873.3 1061.40  4887.4 1058.90  4901.6 1054.88
  4929.8 1046.41  4944.0 1039.36  4958.1 1035.82  4972.3 1033.66  4986.2 1035.39
  5008.2 1034.65  5012.0 1033.66  5012.3 1033.16  5016.2 1033.66  5023.5 1035.50
  5081.3 1039.06  5177.5 1041.21  5189.2 1041.60  5248.2 1047.32  5275.9 1052.58
  5327.8 1064.52  5349.0 1067.46  5377.9 1069.12  5400.9 1073.27  5428.0 1076.16
  5443.4 1080.82  5449.3 1081.38  5458.7 1084.21  5469.3 1086.20  5472.3 1086.20
#Mann=5,-1,0
  4859.1   0.035       0  4986.2    0.07       0  5012.0    0.05       0
  5016.2    0.07       0  5177.5    0.12       0
Bank Sta=5012,5016.2
Exp/Cntr=0.3,0.1

Type RM Length L Ch R = 1,28817,444,444,444
BEGIN DESCRIPTION:
Guadalupe Tributary 36 44.0
END DESCRIPTION:
XS GIS Cut Line= 3
      2199074.99     13853575.01      2199425.00     13853275.00
      2199425.00     13853174.99
#Sta/Elev= 30
  4538.6 1064.27  4560.0 1062.54  4566.6 1060.63  4574.3 1059.76  4580.9 1057.64
  4588.6 1056.38  4595.1 1054.29  4623.7 1047.97  4669.6 1043.38  4715.9 1040.11
  4730.1 1039.87  4779.5 1036.86  4822.3 1035.55  4871.7 1032.14  4943.1 1030.40
  4961.7 1028.32  4971.6 1027.40  4978.2 1025.52  4985.9 1024.70  4994.2 1022.02
  4994.5 1021.52  4998.4 1022.02  5009.6 1022.38  5019.6 1026.72  5029.6 1036.20
  5039.6 1041.04  5059.6 1043.87  5089.6 1050.09  5097.1 1052.28  5099.6 1052.28
#Mann=5,-1,0
  4538.6   0.035       0  4669.6    0.07       0  4961.7    0.12       0
  4994.2    0.05       0  4998.4    0.12       0
Bank Sta=4994.2,4998.4
Exp/Cntr=0.3,0.1

Type RM Length L Ch R = 1,28373,419,419,419
BEGIN DESCRIPTION:
Guadalupe Tributary 36 43.0
END DESCRIPTION:
XS GIS Cut Line= 3
      2199424.99     13853825.01      2199825.00     13853425.00
      2199825.00     13853325.00
#Sta/Elev= 30
  4438.9 1059.45  4467.2 1058.13  4523.8 1053.98  4537.9 1052.39  4566.2 1048.80
  4580.3 1045.87  4594.5 1043.88  4608.6 1041.15  4615.7 1038.93  4636.9 1035.28
  4707.6 1037.18  4735.9 1031.86  4753.8 1030.80  4764.2 1030.19  4820.8 1030.04
  4919.8 1027.45  4962.2 1023.93  4976.3 1019.11  4988.3 1017.28  4988.6 1016.78
  4992.3 1016.78  4992.6 1017.28  5001.1 1019.15  5007.1 1019.15  5014.6 1020.66
  5034.6 1021.22  5044.6 1023.71  5064.6 1032.85  5074.6 1034.52  5104.6 1036.13
#Mann=4,-1,0
  4438.9   0.035       0  4753.8    0.12       0  4988.3    0.05       0
  4992.6    0.12       0
Bank Sta=4988.3,4992.6
Exp/Cntr=0.3,0.1

Type RM Length L Ch R = 1,27954,429,429,429
BEGIN DESCRIPTION:
Guadalupe Tributary 36 42.0
END DESCRIPTION:
XS GIS Cut Line= 3
      2199824.97     13853975.04      2200175.00     13853575.00
      2200275.01     13853174.97
#Sta/Elev= 30
  4484.7 1042.37  4563.0 1036.47  4612.4 1032.05  4633.3 1029.39  4655.1 1028.51
  4669.4 1027.08  4683.6 1024.26  4704.5 1025.99  4761.4 1027.97  4768.1 1027.49
  4789.9 1023.66  4907.4 1021.12  4923.7 1019.89  4938.0 1016.62  4945.5 1015.90
  5006.9 1015.23  5007.2 1014.73  5011.3 1015.23  5012.9 1016.66  5018.8 1016.66
  5026.6 1019.88  5034.3 1024.63  5150.3 1032.96  5222.4 1041.69  5263.6 1044.35
  5315.2 1051.41  5369.3 1056.43  5387.3 1059.89  5410.5 1065.56  5428.6 1067.20
#Mann=4,-1,0
  4484.7   0.035       0  4907.4    0.12       0  5006.9    0.05       0
  5011.3    0.12       0
Bank Sta=5006.9,5011.3
Exp/Cntr=0.3,0.1

Type RM Length L Ch R = 1,27525,445,445,445
BEGIN DESCRIPTION:
Guadalupe Tributary 36 41.0
END DESCRIPTION:
XS GIS Cut Line= 3
      2200124.98     13854075.01      2200525.00     13853775.00
      2200924.97     13853675.01
#Sta/Elev= 30
  4499.8 1026.74  4542.5 1026.51  4602.8 1021.76  4603.5 1021.69  4657.1 1018.26
  4677.9 1020.42  4728.8 1021.97  4761.2 1017.87  4854.8 1015.86  4921.7 1015.51
  4942.5 1010.15  4954.7 1009.65  4955.1 1009.15  4959.5 1009.65  4963.4 1010.84
  5010.1 1010.76  5023.0 1012.93  5064.2 1014.32  5082.3 1013.47  5092.6 1014.72
  5100.3 1018.78  5195.7 1026.77  5224.0 1032.50  5257.5 1035.30  5265.2 1037.84
  5288.4 1041.40  5352.9 1049.60  5360.6 1052.37  5381.2 1056.10  5412.1 1059.13
#Mann=8,-1,0
  4499.8   0.035       0  4602.8   0.094       0  4603.5   0.035       0
  4728.8   0.063       0  4761.2   0.035       0  4854.8    0.12       0
  4954.7    0.05       0  4959.5    0.12       0
Bank Sta=4954.7,4959.5
Exp/Cntr=0.3,0.1

Type RM Length L Ch R = 1,27080,445,445,445
BEGIN DESCRIPTION:
Guadalupe Tributary 36 40.0
END DESCRIPTION:
XS GIS Cut Line= 3
      2200024.96     13854675.03      2200825.00     13854075.00
      2201025.01     13853874.99
#Sta/Elev= 30
  3994.9 1066.34  4023.1 1066.57  4058.5 1060.16  4094.9 1058.72  4202.7 1046.18
  4216.8 1044.91  4237.7 1037.86  4281.4 1033.13  4316.8 1024.64  4352.2 1021.90
  4381.4 1024.18  4441.0 1022.82  4454.7 1022.61  4538.7 1020.71  4637.7 1016.52
  4681.4 1010.76  4749.6 1014.43  4781.4 1010.23  4832.7 1009.74  4981.4 1010.02
  5006.7 1007.39  5007.0 1006.89  5011.5 1007.39  5023.2 1008.38  5051.5 1017.54
  5136.4 1030.15  5164.7 1039.23  5207.1 1044.71  5235.4 1052.63  5277.8 1056.28
#Mann=9,-1,0
  3994.9   0.063       0  4202.7   0.035       0  4441.0   0.094       0
  4454.7   0.035       0  4538.7   0.094       0  4749.6   0.063       0
  4832.7    0.12       0  5006.7    0.05       0  5011.5    0.12       0
Bank Sta=5006.7,5011.5
Exp/Cntr=0.3,0.1

Type RM Length L Ch R = 1,26635,478,478,478
BEGIN DESCRIPTION:
Guadalupe Tributary 36 39.0
END DESCRIPTION:
XS GIS Cut Line= 3
      2200674.98     13854675.01      2201075.00     13854425.00
      2201174.97     13854325.03
#Sta/Elev= 30
  4528.3 1016.69  4557.2 1015.05  4609.1 1010.90  4622.7 1008.73  4630.3 1006.54
  4636.2 1005.68  4658.0 1004.49  4681.6 1003.77  4703.4 1003.72  4724.7 1005.83
  4767.1 1006.68  4797.8 1004.85  4861.5 1002.62  4905.7 1002.39  4949.9 1002.89
  4964.6 1003.50  4971.1 1002.79  4986.7  999.74  4994.7  999.02  4995.0  998.52
  4999.1  998.52  4999.5  999.02  5003.6  999.02  5014.2 1001.38  5028.3 1007.43
  5042.4 1011.55  5084.9 1017.78  5127.3 1027.47  5137.9 1028.75  5141.4 1028.75
#Mann=4,-1,0
  4528.3   0.094       0  4986.7    0.12       0  4994.7    0.05       0
  4999.5    0.12       0
Bank Sta=4994.7,4999.5
Exp/Cntr=0.3,0.1

Type RM Length L Ch R = 1,26157,414,414,414
BEGIN DESCRIPTION:
Guadalupe Tributary 36 38.0
END DESCRIPTION:
XS GIS Cut Line= 3
      2200875.05     13854825.00      2201275.00     13854825.00
      2201475.00     13854525.01
#Sta/Elev= 30
  4595.5 1008.65  4605.5 1008.56  4615.5 1007.17  4655.5 1005.03  4675.5 1002.61
  4695.5 1001.51  4745.5 1002.28  4755.5 1001.59  4805.5 1001.43  4845.5 1000.41
  4990.5  999.99  4990.9  999.49  4995.1  999.49  4995.5  999.99  5003.0 1000.96
  5029.5 1001.98  5096.1 1004.12  5111.1 1003.49  5117.1 1004.43  5126.2 1003.03
  5132.2 1003.95  5147.2 1001.47  5168.2 1002.41  5198.3 1007.37  5234.3 1010.80
  5261.4 1014.67  5276.4 1017.51  5320.0 1027.53  5329.0 1029.02  5356.0 1030.41
#Mann=5,-1,0
  4595.5    0.12       0  4990.5    0.05       0  4995.5    0.12       0
  5029.5   0.063       0  5329.0    0.12       0
Bank Sta=4990.5,4995.5
Exp/Cntr=0.3,0.1

Type RM Length L Ch R = 1,25743,447,447,447
BEGIN DESCRIPTION:
Guadalupe Tributary 36 37.0
END DESCRIPTION:
XS GIS Cut Line= 3
      2201425.01     13855874.97      2201575.00     13855075.00
      2201625.01     13854824.96
#Sta/Elev= 30
  4185.8 1008.33  4236.6 1006.53  4264.6 1003.84  4269.7 1005.00  4287.5 1004.18
  4307.9 1002.24  4328.2  998.46  4409.6  990.55  4485.1  988.90  4552.0  985.29
  4590.2  987.73  4600.4  984.96  4600.8  984.46  4605.4  984.96  4613.1  986.70
  4664.0  989.51  4705.5  989.30  4805.6  992.61  4886.7  991.79  4928.5  990.05
  4959.0  990.40  5020.1  986.62  5030.3  988.96  5081.3  994.04  5162.9  996.39
  5173.1  997.54  5193.5 1010.32  5224.1 1018.04  5236.9 1019.52  5254.7 1020.15
#Mann=5,-1,0
  4185.8   0.035       0  4600.4    0.05       0  4605.4   0.035       0
  4886.7    0.12       0  5236.9   0.094       0
Bank Sta=4600.4,4605.4
Exp/Cntr=0.3,0.1

Type RM Length L Ch R = 1,25296,446,446,446
BEGIN DESCRIPTION:
Guadalupe Tributary 36 36.0
END DESCRIPTION:
XS GIS Cut Line= 3
      2201525.01     13855724.99      2201925.00     13855325.00
      2201975.00     13855025.01
#Sta/Elev= 30
  4429.6  996.11  4457.9  991.49  4483.5  989.41  4500.3  989.34  4514.4  987.79
  4528.6  984.69  4542.7  983.34  4571.0  983.69  4599.3  982.73  4627.6  985.56
  4655.9  986.46  4797.3  987.92  4853.9  986.47  4896.3  987.17  4938.7  985.02
  4967.0  980.88  4981.1  977.69  5002.9  976.57  5003.3  976.07  5007.9  976.57
  5015.6  977.61  5023.2  982.96  5035.8  986.92  5089.1  988.22  5113.9  989.78
  5157.5  990.71  5210.7  993.57  5266.5 1000.81  5274.4 1000.97  5299.4 1003.19
#Mann=6,-1,0
  4429.6   0.035       0  4483.5    0.12       0  5002.9    0.05       0
  5007.9    0.12       0  5113.9   0.035       0  5274.4    0.12       0
Bank Sta=5002.9,5007.9
Exp/Cntr=0.3,0.1

Type RM Length L Ch R = 1,24850,418,418,418
BEGIN DESCRIPTION:
Guadalupe Tributary 36 35.0
END DESCRIPTION:
XS GIS Cut Line= 3
      2201875.03     13855974.97      2202275.00     13855575.00
      2202325.00     13855274.97
#Sta/Elev= 30
  4434.4 1009.89  4437.9 1009.89  4462.6 1001.95  4476.8  995.52  4490.9  990.35
  4505.1  982.55  4519.2  977.16  4547.5  977.19  4618.2  982.39  4674.8  981.01
  4731.3  981.12  4759.6  979.99  4773.8  980.70  4802.0  980.33  4858.6  982.49
  4872.8  981.83  4915.2  977.96  4943.5  977.85  4994.0  971.68  4994.4  971.18
  4999.0  971.68  5050.7  975.14  5060.9  976.60  5111.6  977.10  5142.0  979.10
  5162.2  982.60  5210.4  985.79  5233.2  986.01  5265.5  987.86  5304.2  989.58
#Mann=4,-1,0
  4434.4    0.12       0  4994.0    0.05       0  4999.0    0.12       0
  5265.5   0.035       0
Bank Sta=4994,4999
Exp/Cntr=0.3,0.1

Type RM Length L Ch R = 1,24432,435,435,435
BEGIN DESCRIPTION:
Guadalupe Tributary 36 34.0
END DESCRIPTION:
XS GIS Cut Line= 3
      2202375.01     13856174.98      2202625.00     13855775.00
      2202525.00     13855475.01
#Sta/Elev= 30
  4522.6 1010.56  4551.5 1008.33  4566.8 1002.84  4572.7 1002.45  4588.0  997.77
  4603.4  996.88  4609.3  997.47  4624.6  993.36  4645.8  991.80  4661.1  984.72
  4667.0  984.55  4682.4  977.29  4703.6  973.84  4755.5  970.21  4761.4  970.24
  4776.7  972.99  4813.3  974.65  4834.5  973.62  4913.5  972.81  4958.9  970.51
  4986.6  967.91  4991.3  966.00  4996.9  966.00  5002.3  962.71  5002.7  962.21
  5007.3  962.71  5025.9  967.76  5057.5  968.89  5110.2  973.53  5310.5  979.02
#Mann=3,-1,0
  4522.6    0.12       0  5002.3    0.05       0  5007.3    0.12       0
Bank Sta=5002.3,5007.3
Exp/Cntr=0.3,0.1

Type RM Length L Ch R = 1,23997,466,466,466
BEGIN DESCRIPTION:
Guadalupe Tributary 36 33.0
END DESCRIPTION:
XS GIS Cut Line= 3
      2202625.02     13856474.96      2203025.00     13855675.00
      2202924.99     13855474.99
#Sta/Elev= 30
  4105.6 1036.24  4141.9 1034.56  4172.6 1026.30  4217.4 1026.36  4280.0 1016.01
  4337.5 1013.17  4404.6 1000.68  4432.6  998.58  4477.3  991.43  4494.1  985.56
  4499.7  985.89  4544.4  977.08  4561.2  971.36  4583.5  968.59  4633.8  967.86
  4673.0  970.07  4843.5  969.33  4879.8  968.49  4894.9  965.39  4924.5  962.18
  4969.2  961.34  4983.5  958.54  4983.9  958.04  4988.6  958.54  4991.6  962.78
  4997.2  964.61  5115.4  970.36  5148.1  970.07  5164.9  973.81  5223.6  975.52
#Mann=6,-1,0
  4105.6   0.035       0  4280.0    0.12       0  4894.9   0.035       0
  4983.5   0.035       0  4988.6   0.035       0  5115.4    0.12       0
Bank Sta=4983.5,4988.6
Exp/Cntr=0.3,0.1

Type RM Length L Ch R = 1,23531,480,480,480
BEGIN DESCRIPTION:
Guadalupe Tributary 36 32.0
END DESCRIPTION:
XS GIS Cut Line= 3
      2203001.59     13856638.96      2203475.00     13855625.00
      2203724.97     13855275.04
#Sta/Elev= 30
  3881.0 1024.67  3940.6 1016.65  4021.2 1014.04  4061.4 1008.16  4066.9 1009.99
  4089.8 1004.65  4158.3  996.38  4163.8  998.26  4181.2  994.12  4186.7  995.99
  4204.0  992.13  4209.6  993.79  4255.3  987.54  4292.0  986.22  4434.0  976.79
  4600.1  969.50  4856.6  965.28  4934.4  961.02  4955.9  957.18  4974.3  949.14
  4974.8  948.64  4981.6  949.14  5049.2  957.26  5200.3  961.29  5286.4  967.06
  5322.0  977.60  5366.2  997.60  5393.3 1004.79  5414.9 1006.94  5430.1 1008.46
#Mann=8,-1,0
  3881.0   0.035       0  4292.0    0.12       0  4434.0    0.07       0
  4600.1   0.035       0  4934.4    0.12       0  4974.3    0.05       0
  4981.6    0.12       0  5414.9   0.063       0
Bank Sta=4974.3,4981.6
Exp/Cntr=0.3,0.1

Type RM Length L Ch R = 1,23051,448,448,448
BEGIN DESCRIPTION:
Guadalupe Tributary 36 31.0
END DESCRIPTION:
XS GIS Cut Line= 3
      2203200.03     13856699.96      2203925.00     13855625.00
      2203999.66     13855130.38
#Sta/Elev= 30
  3708.1 1022.48  3744.0 1018.16  3786.5 1017.34  3810.0 1012.25  3967.4 1002.77
  4016.9  997.49  4101.0  983.73  4169.7  982.39  4196.8  975.97  4225.7  973.70
  4377.5  969.48  4449.8  964.07  4643.5  961.33  4709.4  963.87  4766.4  960.46
  4811.3  961.00  4961.2  953.58  4976.2  948.58  4998.0  946.19  4998.5  945.69
  5005.4  946.19  5029.4  955.92  5045.1  964.90  5085.6  982.38  5103.0  992.75
  5126.0 1000.09  5240.8 1004.71  5304.6 1012.62  5411.6 1020.94  5504.9 1026.22
#Mann=7,-1,0
  3708.1   0.035       0  4101.0    0.12       0  4225.7   0.035       0
  4998.0   0.035       0  5005.4   0.035       0  5029.4    0.12       0
  5411.6   0.063       0
Bank Sta=4998,5005.4
Exp/Cntr=0.3,0.1

Type RM Length L Ch R = 1,22603,470,470,470
BEGIN DESCRIPTION:
Guadalupe Tributary 36 30.0
END DESCRIPTION:
XS GIS Cut Line= 3
      2203925.04     13855974.99      2204275.00     13855875.00
      2204375.03     13855824.99
#Sta/Elev= 30
  4636.0  958.45  4667.2  957.81  4691.9  957.99  4725.7  956.63  4798.5  955.24
  4803.7  955.39  4896.0  953.88  4937.6  951.87  4944.1  950.96  4958.4  950.64
  4977.9  948.77  4989.6  945.26  4997.4  944.72  5013.9  944.15  5027.0  943.20
  5027.5  942.70  5034.0  942.70  5034.5  943.20  5036.3  946.26  5044.7  951.17
  5053.1  958.57  5058.7  960.62  5067.0  962.85  5075.4  966.04  5081.0  966.82
  5089.4  970.84  5097.8  974.35  5103.4  973.06  5109.0  974.92  5111.8  974.92
#Mann=3,-1,0
  4636.0   0.035       0  5027.0   0.035       0  5034.5   0.035       0
Bank Sta=5027,5034.5
Exp/Cntr=0.3,0.1

Type RM Length L Ch R = 1,22133,469,469,469
BEGIN DESCRIPTION:
Guadalupe Tributary 36 29.0
END DESCRIPTION:
XS GIS Cut Line= 3
      2204175.00     13856225.00      2204575.00     13856225.00
      2204625.01     13855874.95
#Sta/Elev= 30
  4600.0  955.55  4630.0  955.00  4660.0  953.59  4690.0  953.00  4750.0  952.37
  4780.0  953.09  4810.0  952.92  4860.0  950.65  4880.0  950.18  4910.0  949.74
  4930.0  950.48  4940.0  950.43  4980.0  947.69  4990.0  941.52  4993.7  939.70
  4994.2  939.20  5000.7  939.20  5001.2  939.70  5030.3  941.09  5040.4  945.32
  5060.6  948.23  5070.7  948.52  5090.9  946.89  5121.2  948.04  5191.9  952.00
  5212.1  955.32  5252.5  960.75  5262.6  962.45  5292.9  968.84  5353.6  973.56
#Mann=3,-1,0
  4600.0   0.035       0  4993.7   0.035       0  5001.2   0.035       0
Bank Sta=4993.7,5001.2
Exp/Cntr=0.3,0.1

Type RM Length L Ch R = 1,21664,430,430,430
BEGIN DESCRIPTION:
Guadalupe Tributary 36 28.0
END DESCRIPTION:
XS GIS Cut Line= 3
      2204475.00     13856875.00      2204875.00     13856575.00
      2205075.04     13856524.99
#Sta/Elev= 30
  4504.5  954.36  4568.0  950.24  4726.4  945.17  4754.5  945.28  4761.8  946.57
  4768.0  946.69  4791.0  944.23  4811.8  943.61  4832.6  943.82  4861.8  943.07
  4897.2  943.61  4918.0  946.52  4932.6  946.94  4947.2  945.58  4961.8  941.44
  4986.7  936.22  4987.2  935.72  4994.7  935.72  4995.2  936.22  4997.2  936.93
  5007.1  936.84  5014.8  938.01  5022.5  940.40  5035.4  942.44  5068.9  944.45
  5117.9  949.74  5146.2  951.15  5169.4  951.51  5179.7  952.72  5210.7  952.97
#Mann=3,-1,0
  4504.5   0.035       0  4986.7   0.035       0  4995.2   0.035       0
Bank Sta=4986.7,4995.2
Exp/Cntr=0.3,0.1

Type RM Length L Ch R = 1,21234,581,581,581
BEGIN DESCRIPTION:
Guadalupe Tributary 36 27.0
END DESCRIPTION:
XS GIS Cut Line= 3
      2204299.16     13857139.92      2204875.00     13856975.00
      2205458.03     13856662.48
#Sta/Elev= 30
  4401.1  981.12  4428.0  977.84  4435.2  975.60  4474.5  973.21  4513.1  965.08
  4614.4  953.37  4619.6  954.05  4625.6  951.63  4741.4  947.42  4844.1  941.43
  4949.4  938.98  4978.0  932.93  4983.2  933.68  4985.4  932.19  4985.9  931.69
  4993.9  932.19  5035.8  937.39  5052.1  942.44  5090.3  944.86  5124.9  943.93
  5156.0  948.76  5199.9  945.45  5369.7  948.80  5457.4  952.23  5517.5  957.74
  5536.7  957.53  5567.4  960.50  5577.6  959.78  5612.8  965.17  5661.6  967.92
#Mann=6,-1,0
  4401.1   0.035       0  4474.5    0.12       0  4741.4   0.035       0
  4985.4   0.035       0  4993.9   0.035       0  5536.7    0.12       0
Bank Sta=4985.4,4993.9
Exp/Cntr=0.3,0.1

Type RM Length L Ch R = 1,20653,333,333,333
BEGIN DESCRIPTION:
Guadalupe Tributary 36 26.0
END DESCRIPTION:
XS GIS Cut Line= 3
      2204375.04     13857525.00      2204772.23     13857526.21
      2205492.73     13856827.42
#Sta/Elev= 30
  4599.1 1002.87  4639.1  996.02  4689.1  980.50  4759.1  970.53  4809.1  967.56
  4849.1  962.18  4909.1  949.69  4919.1  945.12  4956.6  934.13  4969.1  930.14
  4990.8  928.12  4991.3  927.62  4999.5  928.12  5013.3  929.79  5034.5  929.77
  5041.6  931.46  5048.6  930.24  5076.9  936.30  5091.0  936.81  5161.8  934.64
  5211.2  937.59  5218.4  939.17  5543.5  943.19  5784.0  947.95  5847.8  952.98
  5911.4  954.79  5925.5  955.89  5942.1  959.65  5976.2  960.56  6000.0  963.76
#Mann=6,-1,0
  4599.1    0.12       0  4956.6   0.035       0  4990.8   0.035       0
  4999.5   0.035       0  5942.1   0.063       0  5976.2    0.12       0
Bank Sta=4990.8,4999.5
Exp/Cntr=0.3,0.1

Type RM Length L Ch R = 1,20320,413,413,413
BEGIN DESCRIPTION:
Guadalupe Tributary 36 25.0
END DESCRIPTION:
XS GIS Cut Line= 3
      2204275.09     13857878.07      2204875.00     13857825.00
      2205657.08     13856933.60
#Sta/Elev= 30
  4402.6 1031.56  4422.6 1026.30  4455.6 1023.34  4502.9 1013.45  4614.4  995.30
  4673.6  985.63  4693.6  980.71  4713.7  972.37  4743.8  972.33  4784.0  967.59
  4833.3  965.64  4874.3  961.96  4948.9  945.47  4978.6  924.11  4980.4  923.34
  4980.9  922.84  4989.1  923.34  5002.3  927.19  5018.6  927.58  5040.4  935.21
  5054.7  936.06  5068.9  933.77  5083.1  936.30  5175.2  934.32  5522.5  941.61
  5578.5  938.55  5614.5  943.08  5841.3  947.00  6002.7  954.47  6190.7  963.04
#Mann=8,-1,0
  4402.6   0.063       0  4455.6    0.12       0  4614.4   0.063       0
  4833.3    0.12       0  4978.6   0.035       0  4980.4   0.035       0
  4989.1   0.035       0  6002.7   0.063       0
Bank Sta=4980.4,4989.1
Exp/Cntr=0.3,0.1

Type RM Length L Ch R = 1,19907,464,464,464
BEGIN DESCRIPTION:
Guadalupe Tributary 36 24.0
END DESCRIPTION:
XS GIS Cut Line= 3
      2204650.10     13858211.40      2205125.00     13858125.00
      2206025.14     13856753.03
#Sta/Elev= 30
  4527.6  973.73  4664.7  964.31  4828.5  947.87  4959.5  936.77  4978.5  931.46
  4983.6  926.79  4990.0  924.39  5003.4  923.51  5003.9  923.01  5012.2  923.51
  5019.4  923.76  5090.2  931.38  5436.8  936.97  5494.0  940.85  5587.4  941.43
  5653.8  947.14  5674.9  946.90  5680.9  944.43  5696.0  943.55  5711.0  943.81
  5732.1  947.75  5783.4  944.72  5840.6  946.27  5855.7  948.48  5913.0  946.99
  6130.0  953.84  6223.4  954.20  6425.3  960.36  6480.1  964.07  6651.2  968.98
#Mann=6,-1,0
  4527.6   0.035       0  4828.5    0.12       0  5003.4    0.05       0
  5012.2    0.12       0  5019.4   0.035       0  6480.1    0.12       0
Bank Sta=5003.4,5012.2
Exp/Cntr=0.3,0.1

Type RM Length L Ch R = 1,19443,443,443,443
BEGIN DESCRIPTION:
Guadalupe Tributary 36 23.0
END DESCRIPTION:
XS GIS Cut Line= 3
      2204795.94     13858433.62      2205425.00     13858425.00
      2206254.31     13857662.77
#Sta/Elev= 30
  4370.9  964.53  4439.2  963.16  4460.0  959.15  4530.0  954.39  4550.0  949.80
  4670.0  938.06  4700.0  933.11  4790.0  930.86  4830.0  934.60  4860.0  929.59
  4953.3  925.11  4985.3  919.92  4985.8  919.42  4994.8  919.92  4997.5  921.71
  5021.3  920.99  5028.1  924.35  5156.7  926.54  5190.8  924.37  5325.9  931.84
  5632.1  939.01  5679.2  941.28  5735.9  947.64  5792.6  958.88  5814.2  966.35
  5863.5  976.36  5976.9  995.97  6061.4 1004.38  6098.0 1005.12  6126.4 1006.16
#Mann=8,-1,0
  4370.9   0.063       0  4439.2   0.035       0  4953.3    0.07       0
  4985.3    0.05       0  4994.8    0.07       0  5156.7   0.035       0
  5632.1    0.12       0  6098.0   0.063       0
Bank Sta=4985.3,4994.8
Exp/Cntr=0.3,0.1

Type RM Length L Ch R = 1,19000,433,433,433
BEGIN DESCRIPTION:
Guadalupe Tributary 36 22.0
END DESCRIPTION:
XS GIS Cut Line= 3
      2204874.95     13858674.99      2205675.00     13858775.00
      2206075.02     13858675.00
#Sta/Elev= 30
  4199.1  960.43  4219.2  958.39  4279.8  952.92  4289.8  950.58  4340.2  948.27
  4360.4  943.37  4420.9  936.63  4511.6  931.21  4592.2  927.72  4763.5  924.43
  4801.3  925.66  4824.0  930.00  4834.0  929.87  4874.4  921.97  4970.3  915.41
  4970.8  914.91  4979.9  915.41  5002.9  919.15  5064.6  923.13  5113.1  923.37
  5180.6  923.89  5193.5  926.58  5215.5  935.30  5270.4  959.65  5294.0  968.44
  5317.2  971.64  5335.2  977.79  5366.1  992.45  5394.5 1000.77  5417.7 1004.98
#Mann=7,-1,0
  4199.1   0.094       0  4219.2   0.035       0  4970.3   0.035       0
  4979.9   0.035       0  5113.1    0.12       0  5215.5   0.094       0
  5270.4    0.12       0
Bank Sta=4970.3,4979.9
Exp/Cntr=0.3,0.1

Type RM Length L Ch R = 1,18567,466,466,466
BEGIN DESCRIPTION:
Guadalupe Tributary 36 21.0
END DESCRIPTION:
XS GIS Cut Line= 3
      2204309.83     13858635.00      2205775.00     13859175.00
      2206074.99     13859175.00
#Sta/Elev= 30
  3438.4  992.93  3441.9  992.81  3481.5  986.75  3658.8  973.43  3771.6  969.19
  3916.8  961.25  4088.9  955.47  4136.7  956.51  4195.4  947.85  4276.8  945.73
  4291.3  940.26  4296.6  942.29  4355.1  930.56  4499.1  923.89  4690.8  921.39
  4721.3  923.52  4797.4  919.60  4936.0  918.75  4991.2  914.17  5015.1  913.36
  5015.6  912.86  5024.8  913.36  5039.9  917.68  5099.9  923.20  5179.9  961.35
  5199.9  974.44  5226.0  976.12  5239.9  978.56  5253.3  985.20  5299.9 1001.01
#Mann=11,-1,0
  3438.4   0.094       0  3441.9   0.035       0  3771.6   0.094       0
  4195.4   0.035       0  4276.8   0.094       0  4355.1   0.035       0
  4991.2    0.12       0  5015.1    0.05       0  5024.8    0.12       0
  5226.0   0.035       0  5253.3    0.12       0
Bank Sta=5015.1,5024.8
Exp/Cntr=0.3,0.1

Type RM Length L Ch R = 1,18101,439,439,439
BEGIN DESCRIPTION:
Guadalupe Tributary 36 20.0
END DESCRIPTION:
XS GIS Cut Line= 3
      2203386.27     13858253.09      2205725.00     13859625.00
      2206031.04     13859503.47
#Sta/Elev= 30
  2288.2 1051.63  2388.1 1052.43  2533.9 1049.14  2676.2 1041.06  2873.6 1023.16
  2895.1 1017.39  3011.1 1009.79  3082.1 1002.76  3116.1 1000.20  3246.9  990.77
  3318.5  979.55  3350.8  979.77  3567.3  964.91  3878.9  954.83  4137.9  942.21
  4304.0  926.57  4516.7  918.73  4656.8  917.78  4807.2  916.89  4970.3  913.58
  4986.9  909.41  4987.4  908.91  4996.6  909.41  5068.5  914.59  5092.8  928.15
  5122.4  934.56  5171.1  954.49  5257.8  963.21  5284.4  965.36  5328.9  978.46
#Mann=14,-1,0
  2288.2    0.12       0  2388.1   0.063       0  2533.9    0.12       0
  3011.1   0.035       0  3082.1    0.12       0  3116.1   0.035       0
  3350.8   0.094       0  3878.9   0.035       0  4516.7    0.12       0
  4656.8   0.035       0  4807.2    0.12       0  4986.9    0.05       0
  4996.6    0.12       0  5257.8   0.035       0
Bank Sta=4986.9,4996.6
Exp/Cntr=0.3,0.1

Type RM Length L Ch R = 1,17662,451,451,451
BEGIN DESCRIPTION:
Guadalupe Tributary 36 19.0
END DESCRIPTION:
XS GIS Cut Line= 3
      2203400.16     13860648.89      2205675.00     13860025.00
      2205975.00     13859725.00
#Sta/Elev= 30
  2640.6 1006.52  2747.0 1007.90  2894.5 1003.69  3093.4  995.69  3195.2  983.80
  3277.8  982.85  3395.0  977.06  3429.4  972.51  3568.5  968.73  3682.5  958.61
  3786.2  956.86  3805.0  952.98  3832.2  950.40  3935.3  940.71  4086.9  935.37
  4140.3  928.90  4244.3  924.44  4418.8  913.36  4628.6  909.40  4789.2  908.90
  4895.7  912.06  4991.9  908.71  4992.4  908.21  5001.7  908.71  5016.2  909.46
  5027.7  911.93  5197.4  912.98  5254.0  922.53  5353.0  944.62  5423.7  950.74
#Mann=11,-1,0
  2640.6    0.12       0  3277.8   0.035       0  3805.0   0.063       0
  3832.2    0.12       0  3935.3   0.035       0  4140.3    0.12       0
  4244.3    0.07       0  4628.6   0.033       0  4991.9   0.033       0
  5001.7   0.033       0  5016.2    0.12       0
Bank Sta=4991.9,5001.7
Exp/Cntr=0.3,0.1

Type RM Length L Ch R = 1,17211,452,452,452
BEGIN DESCRIPTION:
Guadalupe Tributary 36 18.0
END DESCRIPTION:
XS GIS Cut Line= 3
      2205074.97     13861025.02      2205875.00     13860275.00
      2206240.19     13859524.34
#Sta/Elev= 30
  3908.0  966.01  3936.1  964.85  3971.1  957.95  4017.4  951.21  4042.6  946.91
  4110.1  939.47  4139.8  936.61  4176.9  930.60  4205.3  923.28  4226.3  921.00
  4268.8  908.97  4325.1  909.09  4537.9  909.98  4566.0  908.60  4977.7  908.38
  4978.2  907.88  4989.0  908.38  5137.7  913.71  5282.6  918.38  5327.1  923.13
  5375.6  932.19  5416.1  940.00  5447.1  943.18  5638.6  954.62  5655.6  957.18
  5688.8  959.10  5728.8  964.96  5768.4  977.53  5822.6  984.57  5839.4  986.01
#Mann=12,-1,0
  3908.0   0.063       0  3971.1    0.12       0  4017.4   0.035       0
  4110.1    0.12       0  4139.8   0.035       0  4325.1   0.033       0
  4977.7   0.033       0  4989.0   0.033       0  5137.7    0.12       0
  5375.6   0.035       0  5688.8    0.12       0  5822.6   0.035       0
Bank Sta=4977.7,4989
Exp/Cntr=0.3,0.1

Type RM Length L Ch R = 1,16759,475,475,475
BEGIN DESCRIPTION:
Guadalupe Tributary 36 17.0
END DESCRIPTION:
XS GIS Cut Line= 3
      2203816.79     13862121.12      2206275.00     13860325.00
      2206455.68     13859600.26
#Sta/Elev= 30
  1955.1 1003.73  2123.3  983.97  2262.5  974.86  2440.2  965.00  2531.0  958.23
  2586.2  959.48  2631.4  955.86  2731.8  957.11  2814.6  962.42  2959.7  965.87
  3126.0  959.09  3210.6  955.41  3286.2  959.34  3313.7  960.18  3438.5  960.51
  3446.4  958.59  3563.3  956.00  3603.7  955.53  3810.3  937.75  3911.1  928.48
  3976.0  909.49  4013.4  909.02  4990.6  908.51  4991.1  908.01  5002.3  908.51
  5057.8  911.80  5264.5  937.82  5533.3  954.73  5642.0  961.98  5746.5  982.97
#Mann=18,-1,0
  1955.1   0.035       0  2262.5    0.12       0  2440.2   0.063       0
  2586.2   0.035       0  2814.6    0.12       0  3126.0   0.035       0
  3286.2    0.12       0  3313.7   0.035       0  3438.5    0.12       0
  3446.4   0.035       0  3563.3    0.12       0  3810.3   0.035       0
  4013.4   0.033       0  4990.6   0.033       0  5002.3   0.033       0
  5057.8    0.07       0  5264.5    0.12       0  5533.3   0.035       0
Bank Sta=4990.6,5002.3
Exp/Cntr=0.3,0.1

Type RM Length L Ch R = 1,16284,1348,1348,1348
BEGIN DESCRIPTION:
Guadalupe Tributary 36 16.0
END DESCRIPTION:
XS GIS Cut Line= 3
      2205754.27     13862183.66      2206725.00     13860325.00
      2206608.57     13858948.80
#Sta/Elev= 30
  2913.1  981.13  3164.3  978.60  3202.8  971.60  3379.4  959.84  3395.9  955.00
  3467.8  949.52  3498.2  942.91  3565.9  941.77  3660.9  932.57  3682.9  926.87
  3697.8  915.72  3712.6  910.66  3834.3  911.24  4959.0  908.41  4959.5  907.91
  4970.8  908.41  5062.9  915.23  5210.7  924.22  5351.2  938.84  5422.3  949.63
  5521.8  960.18  5592.1  963.69  5653.2  977.36  5672.3  983.68  5808.1  998.34
  5954.6 1013.72  5983.5 1021.41  6080.8 1032.52  6284.5 1046.52  6391.1 1049.31
#Mann=12,-1,0
  2913.1    0.12       0  3498.2   0.063       0  3697.8    0.07       0
  3834.3   0.033       0  4959.0   0.033       0  4970.8   0.033       0
  5062.9    0.12       0  5422.3   0.063       0  5653.2   0.035       0
  5808.1    0.12       0  5954.6   0.035       0  6080.8    0.12       0
Bank Sta=4959,4970.8
Exp/Cntr=0.3,0.1

Type RM Length L Ch R = 1,14936,468,468,468
BEGIN DESCRIPTION:
Guadalupe Tributary 36 15.0
END DESCRIPTION:
XS GIS Cut Line= 3
      2206025.01     13861874.99      2207825.00     13860225.00
      2208504.28     13859641.96
#Sta/Elev= 30
  2562.9  970.64  2640.9  967.15  2647.7  963.48  2732.8  955.94  2810.5  942.63
  2863.7  939.74  2913.9  935.56  2980.6  930.27  3015.8  920.88  3058.3  919.18
  3079.3  912.99  3145.7  910.97  3170.3  912.62  3235.3  908.98  3292.0  911.51
  4956.0  908.33  4956.5  907.83  4969.0  908.33  5032.7  909.59  5095.9  927.97
  5253.3  961.38  5316.9  969.25  5376.7  969.09  5510.0  975.56  5522.2  975.65
  5565.0  988.65  5657.1 1000.63  5709.2 1002.47  5792.1 1008.55  5899.9 1009.97
#Mann=11,-1,0
  2562.9    0.12       0  2863.7   0.063       0  2913.9   0.035       0
  3145.7    0.07       0  3170.3   0.033       0  4956.0   0.033       0
  4969.0   0.033       0  5095.9    0.12       0  5376.7   0.063       0
  5510.0   0.035       0  5709.2    0.12       0
Bank Sta=4956,4969
Exp/Cntr=0.3,0.1

Type RM Length L Ch R = 1,14468,881,881,881
BEGIN DESCRIPTION:
Guadalupe Tributary 36 14.0
END DESCRIPTION:
XS GIS Cut Line= 3
      2206324.99     13861775.01      2208125.00     13860575.00
      2208427.66     13859899.44
#Sta/Elev= 30
  2840.6  947.31  2854.1  943.94  2899.2  936.51  2905.8  938.02  2935.3  938.11
  2956.3  933.66  3002.6  930.44  3070.5  922.44  3187.6  914.07  3229.7  909.07
  3294.8  908.53  5011.8  908.38  5012.3  907.88  5024.8  908.38  5036.0  910.42
  5047.8  915.42  5070.1  921.36  5103.9  929.05  5124.5  935.18  5157.4  941.42
  5191.5  951.50  5246.4  962.93  5307.5  967.58  5459.1  972.93  5519.0  974.76
  5565.5  986.74  5579.0  989.33  5607.6  997.71  5671.7 1000.35  5744.2 1005.79
#Mann=10,-1,0
  2840.6    0.12       0  2905.8   0.063       0  3002.6   0.035       0
  3294.8   0.033       0  5011.8   0.033       0  5024.8   0.033       0
  5103.9    0.12       0  5246.4   0.063       0  5459.1   0.035       0
  5565.5    0.12       0
Bank Sta=5011.8,5024.8
Exp/Cntr=0.3,0.1

Type RM Length L Ch R = 1,13587,1794,1794,1794
BEGIN DESCRIPTION:
Guadalupe Tributary 36 13.0
END DESCRIPTION:
XS GIS Cut Line= 3
      2206174.98     13861975.01      2207975.00     13861375.00
      2208712.62     13859503.07
#Sta/Elev= 30
  3099.3  972.66  3268.0  967.07  3414.1  948.11  3447.2  940.58  3521.0  940.07
  3549.2  934.77  3615.8  930.79  3647.4  926.71  3658.0  921.80  3862.3  908.44
  3862.8  907.94  3875.3  908.44  3890.4  908.44  5769.6  908.75  5781.3  909.33
  5845.4  927.60  5961.8  957.96  6089.4  967.19  6136.5  968.16  6298.5  974.39
  6340.2  976.31  6361.7  984.87  6403.0  994.76  6427.5  998.21  6562.8 1006.49
  6587.2 1006.95  6592.6 1004.28  6630.4 1009.15  6821.0 1010.42  7008.7 1008.66
#Mann=13,-1,0
  3099.3    0.12       0  3414.1   0.063       0  3549.2   0.035       0
  3862.3   0.033       0  3875.3   0.035       0  3890.4   0.033       0
  5845.4    0.12       0  6089.4   0.063       0  6136.5   0.035       0
  6298.5   0.063       0  6403.0    0.12       0  6427.5   0.035       0
  6821.0    0.12       0
Bank Sta=3862.3,3875.3
Exp/Cntr=0.3,0.1

Type RM Length L Ch R = 1,11793,442,442,442
BEGIN DESCRIPTION:
Guadalupe Tributary 36 12.0
END DESCRIPTION:
XS GIS Cut Line= 3
      2206224.98     13862025.01      2209225.00     13861125.00
      2211330.38     13860530.93
#Sta/Elev= 30
  1859.6  973.16  1995.3  968.50  2037.1  961.62  2116.8  956.28  2232.8  940.76
  2392.1  930.11  2444.3  920.39  2507.3  916.28  2635.9  908.70  3962.5  908.40
  3963.0  907.90  3976.3  908.40  5095.6  908.57  5155.1  924.41  5241.2  938.60
  5333.2  957.86  5539.8  974.17  5638.6  983.38  5706.6  998.90  5746.3 1001.80
  5874.9 1015.96  5947.3 1028.16  6004.6 1029.99  6124.3 1044.94  6345.5 1056.35
  6553.0 1068.99  6725.5 1070.58  6729.5 1070.79  6960.4 1071.73  7179.3 1064.62
#Mann=17,-1,0
  1859.6    0.12       0  2116.8   0.063       0  2232.8   0.035       0
  2507.3    0.07       0  2635.9   0.033       0  3962.5   0.033       0
  3976.3   0.033       0  5241.2   0.035       0  5333.2   0.063       0
  5539.8    0.12       0  5746.3   0.035       0  5947.3    0.12       0
  6345.5   0.063       0  6553.0   0.035       0  6725.5   0.063       0
  6729.5   0.035       0  6960.4   0.063       0
Bank Sta=3962.5,3976.3
Exp/Cntr=0.3,0.1

Type RM Length L Ch R = 1,11351,1089,1089,1089
BEGIN DESCRIPTION:
Guadalupe Tributary 36 11.0
END DESCRIPTION:
XS GIS Cut Line= 3
      2206274.97     13862075.01      2209275.00     13861475.00
      2209825.03     13861124.98
#Sta/Elev= 30
  1944.5  973.00  2015.9  966.09  2026.1  967.37  2148.5  959.10  2209.7  950.76
  2243.3  949.96  2260.7  949.15  2291.3  940.85  2309.1  940.24  2332.1  940.15
  2393.2  932.53  2479.9  928.76  2505.4  926.38  2536.0  919.01  2636.5  913.21
  2723.8  908.68  3844.7  908.38  3845.2  907.88  3858.5  908.38  5205.4  908.58
  5235.9  919.99  5324.6  940.99  5351.1  946.02  5381.5  957.42  5395.1  959.62
  5552.7  972.46  5562.8  973.99  5596.6  978.17  5627.1  989.11  5655.9  989.77
#Mann=10,-1,0
  1944.5    0.12       0  2243.3   0.063       0  2309.1   0.035       0
  2636.5    0.07       0  2723.8   0.033       0  3844.7   0.033       0
  3858.5   0.033       0  5324.6   0.063       0  5552.7   0.035       0
  5562.8   0.063       0
Bank Sta=3844.7,3858.5
Exp/Cntr=0.3,0.1

Type RM Length L Ch R = 1,10262,703,703,703
BEGIN DESCRIPTION:
Guadalupe Tributary 36 10.0
END DESCRIPTION:
XS GIS Cut Line= 3
      2207636.27     13862961.37      2208733.46     13862211.40
      2209920.52     13861225.65
#Sta/Elev= 30
  3678.6  965.62  3725.5  963.66  3739.5  961.73  3819.6  953.82  3861.5  952.06
  3897.4  942.86  3933.3  944.06  4051.0  937.49  4169.0  932.78  4222.1  928.70
  4271.2  921.25  4301.1  919.12  4444.6  911.85  4474.5  908.86  4515.7  908.68
  5190.8  908.48  5191.3  907.98  5205.0  908.48  6085.9  909.34  6149.7  931.77
  6185.1  941.81  6248.7  956.62  6283.8  960.78  6304.5  961.55  6316.5  962.04
  6348.5  963.41  6376.3  968.88  6433.6  973.91  6490.9  988.19  6550.6  995.21
#Mann=10,-1,0
  3678.6    0.12       0  3739.5   0.063       0  4051.0    0.12       0
  4169.0   0.035       0  4515.7   0.033       0  5190.8   0.033       0
  5205.0   0.033       0  6185.1   0.035       0  6304.5   0.063       0
  6316.5   0.035       0
Bank Sta=5190.8,5205
Exp/Cntr=0.3,0.1

Type RM Length L Ch R = 1,9559,447,447,447
BEGIN DESCRIPTION:
Guadalupe Tributary 36 9.0
END DESCRIPTION:
XS GIS Cut Line= 3
      2207698.71     13863003.07      2208525.00     13862675.00
      2210324.99     13861175.01
#Sta/Elev= 30
  4111.9  963.01  4135.5  962.17  4200.4  954.43  4278.8  951.39  4323.1  942.14
  4457.7  937.08  4624.4  929.37  4708.9  919.31  4860.8  909.79  6484.9  908.55
  6485.4  908.05  6499.1  908.55  6627.4  909.32  6633.9  913.23  6648.2  914.63
  6654.8  921.08  6683.4  933.12  6712.1  938.12  6839.6  960.05  6946.3  969.03
  6960.7  967.65  7102.5  984.06  7109.7  984.34  7116.9  980.13  7123.4  983.29
  7131.2  980.71  7137.7  985.69  7145.5  983.86  7223.6 1007.85  7344.0 1029.56
#Mann=8,-1,0
  4111.9    0.12       0  4135.5   0.063       0  4457.7   0.035       0
  4708.9    0.07       0  4860.8   0.033       0  6484.9   0.033       0
  6499.1   0.033       0  6712.1    0.12       0
Bank Sta=6484.9,6499.1
Exp/Cntr=0.3,0.1

Type RM Length L Ch R = 1,9112,928,928,928
BEGIN DESCRIPTION:
Guadalupe Tributary 36 8.0
END DESCRIPTION:
XS GIS Cut Line= 3
      2207726.47     13863079.46      2208775.00     13862875.00
      2210575.03     13861074.97
#Sta/Elev= 30
  3931.3  961.80  4001.1  953.77  4024.0  953.52  4103.0  949.25  4133.0  942.28
  4225.9  939.16  4448.4  927.80  4530.9  918.03  4629.9  913.18  4730.9  908.60
  4863.4  908.23  4863.9  907.73  4877.7  908.23  6696.6  908.51  6724.9  908.60
  6767.3  912.19  6823.9  908.87  6880.5  917.01  6894.6  921.36  6920.4  934.59
  6951.2  952.08  6979.5  961.65  7064.3  975.36  7135.0  992.12  7177.5  998.69
  7347.2 1032.56  7357.8 1034.33  7417.9 1043.53  7517.7 1048.59  7545.2 1049.73
#Mann=12,-1,0
  3931.3   0.094       0  4024.0   0.063       0  4225.9    0.07       0
  4448.4   0.035       0  4629.9    0.07       0  4730.9   0.033       0
  4863.4   0.033       0  4877.7   0.033       0  6920.4    0.12       0
  7347.2   0.063       0  7357.8   0.035       0  7517.7   0.063       0
Bank Sta=4863.4,4877.7
Exp/Cntr=0.3,0.1

Type RM Length L Ch R = 1,8184,950,950,950
BEGIN DESCRIPTION:
Guadalupe Tributary 36 7.0
END DESCRIPTION:
XS GIS Cut Line= 3
      2207028.07     13863786.88      2209675.00     13862875.00
      2210674.97     13861675.04
#Sta/Elev= 30
  2200.4 1046.38  2228.9 1039.12  2285.0 1030.75  2355.8 1016.02  2409.9 1008.33
  2535.6  983.82  2813.0  958.20  2893.4  950.83  2948.1  948.60  3018.3  941.36
  3221.2  934.00  3297.4  930.22  3521.0  926.35  3600.8  917.46  3652.6  914.92
  3757.9  910.36  3812.2  908.30  3812.7  907.80  3826.5  908.30  6271.1  908.66
  6277.6  909.44  6310.4  922.56  6349.2  939.45  6370.0  953.65  6384.4  959.18
  6405.8  958.63  6456.0  969.14  6511.9  974.02  6522.2  980.97  6562.0  990.59
#Mann=11,-1,0
  2200.4    0.12       0  2813.0   0.094       0  3221.2   0.035       0
  3297.4    0.07       0  3521.0   0.035       0  3652.6    0.07       0
  3757.9   0.033       0  3812.2   0.033       0  3826.5   0.033       0
  6310.4    0.12       0  6522.2   0.035       0
Bank Sta=3812.2,3826.5
Exp/Cntr=0.3,0.1

Type RM Length L Ch R = 1,7234,962,962,962
BEGIN DESCRIPTION:
Guadalupe Tributary 36 6.0
END DESCRIPTION:
XS GIS Cut Line= 3
      2207092.66     13863895.48      2210625.00     13862875.00
      2210974.99     13862275.02
#Sta/Elev= 30
  1323.2 1038.59  1342.1 1035.01  1388.1 1030.90  1448.2 1018.89  1520.7 1009.59
  1525.9 1010.65  1554.3 1004.61  1581.5 1002.27  1618.7  997.64  1738.0  978.01
  1926.7  955.80  1960.6  951.27  2027.9  947.33  2033.4  944.52  2061.5  941.04
  2122.8  938.27  2324.9  929.41  2351.4  925.78  2457.4  919.72  2575.2  915.67
  2678.7  911.83  2740.1  908.23  2740.6  907.73  2754.4  908.23  5461.8  909.16
  5483.3  910.79  5504.8  916.53  5547.8  919.81  5585.1  925.44  5694.6  937.56
#Mann=10,-1,0
  1323.2    0.12       0  1581.5   0.033       0  1618.7    0.12       0
  1926.7   0.094       0  2122.8   0.035       0  2575.2    0.07       0
  2678.7   0.033       0  2740.1   0.033       0  2754.4   0.033       0
  5585.1    0.07       0
Bank Sta=2740.1,2754.4
Exp/Cntr=0.3,0.1

Type RM Length L Ch R = 1,6272,464,464,464
BEGIN DESCRIPTION:
Guadalupe Tributary 36 5.0
END DESCRIPTION:
XS GIS Cut Line= 3
      2209420.56     13865680.71      2211525.00     13862975.00
      2211774.99     13862725.01
#Sta/Elev= 30
  1583.2  908.00  1583.7  907.50  1597.7  908.00  2337.9  908.91  2346.0  909.30
  2352.4  910.82  2360.5  918.77  2364.3  919.27  2375.0  920.14  2410.3  917.71
  2451.9  916.39  2495.3  913.78  2524.3  910.91  2530.6  911.29  2538.8  909.14
  2586.5  908.93  2887.2  910.10  3749.5  908.42  4997.4  908.31  5014.5  908.50
  5039.2  910.42  5067.5  916.16  5090.7  919.03  5110.0  921.39  5166.5  930.72
  5194.8  932.33  5237.2  937.44  5265.5  942.96  5322.1  951.38  5364.5  953.02
#Mann=5,-1,0
  1583.2   0.033       0  1597.7   0.033       0  2364.3   0.035       0
  2586.5   0.033       0  5090.7   0.063       0
Bank Sta=1583.2,1597.7
Exp/Cntr=0.3,0.1

Type RM Length L Ch R = 1,5808,875,875,875
BEGIN DESCRIPTION:
Guadalupe Tributary 36 4.0
END DESCRIPTION:
XS GIS Cut Line= 3
      2209770.84     13865980.95      2211875.00     13862975.00
      2211975.01     13862724.98
#Sta/Elev= 30
  1321.8  908.00  1322.3  907.50  1336.4  908.00  1946.8  908.83  1952.9  909.49
  1976.0  920.14  1995.1  922.65  2012.2  922.83  2091.0  917.29  2161.3  913.76
  2190.9  913.73  2211.9  911.04  2230.3  910.70  2270.6  910.74  5059.7  908.71
  5077.2  912.78  5083.9  918.90  5089.3  918.06  5108.2  925.10  5113.5  924.68
  5131.0  931.66  5137.8  935.85  5143.2  935.45  5151.1  937.88  5162.0  941.93
  5167.4  941.75  5191.6  950.77  5221.2  956.55  5245.5  967.22  5260.3  967.77
#Mann=7,-1,0
  1321.8   0.033       0  1336.4   0.033       0  1995.1    0.07       0
  2091.0   0.035       0  2230.3    0.07       0  2270.6   0.033       0
  5151.1    0.12       0
Bank Sta=1321.8,1336.4
Exp/Cntr=0.3,0.1

Type RM Length L Ch R = 1,4933,438,438,438
BEGIN DESCRIPTION:
Guadalupe Tributary 36 3.0
END DESCRIPTION:
XS GIS Cut Line= 3
      2211372.04     13865831.67      2212575.00     13863125.00
      2212525.00     13862575.02
#Sta/Elev= 30
  2038.6  908.00  2039.1  907.50  2052.7  907.50  2053.2  908.00  4956.8  908.00
  4991.7  908.75  5060.8  911.37  5151.2  913.60  5161.2  910.79  5171.3  909.24
  5231.5  911.43  5241.5  911.02  5271.7  923.94  5306.4  941.28  5342.0  959.90
  5352.0  963.47  5362.0  967.93  5372.1  971.43  5380.9  973.46  5402.2  981.58
  5412.2  987.24  5432.3  994.49  5442.4  997.37  5452.4 1002.49  5462.5 1005.92
  5492.6 1013.95  5502.6 1018.23  5512.7 1020.50  5550.3 1031.12  5552.8 1031.12
#Mann=4,-1,0
  2038.6   0.033       0  2053.2   0.033       0  5306.4    0.07       0
  5380.9    0.12       0
Bank Sta=2038.6,2053.2
Exp/Cntr=0.3,0.1

Type RM Length L Ch R = 1,4495,917,917,917
BEGIN DESCRIPTION:
Guadalupe Tributary 36 2.0
END DESCRIPTION:
XS GIS Cut Line= 3
      2211371.45     13865981.39      2212875.00     13863275.00
      2212990.20     13862345.00
#Sta/Elev= 30
  1892.9  908.00  1893.4  907.50  1907.6  908.00  5472.6  908.40  5482.6  910.76
  5492.7  918.38  5512.8  925.76  5517.8  926.57  5522.9  929.76  5543.1  936.84
  5567.8  947.36  5583.4  953.56  5598.8  961.44  5613.6  962.91  5633.8  968.30
  5643.9  972.29  5664.0  976.57  5674.1  979.79  5679.7  983.76  5744.6 1005.78
  5754.7 1008.53  5760.7 1011.83  5774.9 1016.49  5784.9 1022.14  5795.0 1026.24
  5806.0 1032.65  5825.2 1033.31  5865.5 1041.49  5904.7 1046.07  5926.0 1047.00
#Mann=5,-1,0
  1892.9   0.033       0  1907.6   0.033       0  5567.8    0.12       0
  5806.0   0.063       0  5904.7   0.094       0
Bank Sta=1892.9,1907.6
Exp/Cntr=0.3,0.1

Type RM Length L Ch R = 1,3578,0,0,0
BEGIN DESCRIPTION:
Guadalupe Tributary 36 1.0
END DESCRIPTION:
XS GIS Cut Line= 3
      2212071.45     13865731.39      2213575.00     13863025.00
      2213475.00     13862424.98
#Sta/Elev= 30
  1904.0  908.00  1904.5  907.50  1918.2  907.50  1918.7  908.00  5202.8  908.00
  5263.6  908.89  5276.3  910.87  5283.9  918.12  5329.5  936.60  5332.0  938.21
  5337.1  938.45  5344.7  943.39  5352.6  946.97  5385.2  961.64  5392.8  967.09
  5415.7  971.03  5425.8  976.85  5435.9  979.67  5446.1  980.41  5453.7  982.13
  5458.7  981.38  5476.5  984.66  5486.6  990.30  5506.9  998.62  5514.5 1002.85
  5519.6 1002.91  5547.4 1013.27  5588.0 1023.46  5598.1 1025.29  5608.3 1025.41
#Mann=3,-1,0
  1904.0   0.033       0  1918.7   0.033       0  5352.6    0.12       0
Bank Sta=1904,1918.7
Exp/Cntr=0.3,0.1

Chan Stop Cuts=-1
