--- Miller Creek.prj (project) ---

Proj Title=Miller Creek Base Level Engineering
Current Plan=p01
Default Exp/Contr=0.3,0.1
English Units
Geom File=g01
Flow File=f01
Plan File=p01
BEGIN DESCRIPTION:
Miller Creek
END DESCRIPTION:

--- Miller Creek.p01 (plan) ---

Plan Title=Multiple Run
Short Identifier=Multiple
Geom File=g01
Flow File=f01
Subcritical Flow
K Sum by GR= 0
Std Step Tol= 0.01
Critical Tol= 0.01
Num of Std Step Trials= 20
Max Error Tol= 0.3
Flow Tol Ratio= 0.001
Split Flow NTrial= 30
Split Flow Tol= 0.02
Split Flow Ratio= 0.02
Log Output Level= 0
Friction Slope Method= 1
Unsteady Friction Slope Method= 2
Unsteady Bridges Friction Slope Method= 1
Parabolic Critical Depth
Global Vel Dist=  1 , 1 , 1
Global Log Level= 0
CheckData=True
Encroach Param= -1, 0, 0, 0
BEGIN DESCRIPTION:
Multiple Run
END DESCRIPTION:

--- Miller Creek.f01 (steady flow) ---

Flow Title=Multiple
Number of Profiles=7
Profile Names=10-year,25-year,50-year,1pct_min,100-year,1pct_plu,500-year
River Rch & RM= Miller Creek,Reach-1,20856
    1797    3137    4445    3046    6078   12128   11257
River Rch & RM= Miller Creek,Reach-1,18714
    2107    3703    5272    3627    7237   14439   13511
River Rch & RM= Miller Creek,Reach-1,14634
    2990    5324    7642    5294   10563   21075   20000
River Rch & RM= Miller Creek,Reach-1,6905
    4429    7999   11596    8101   16165   32253   31133
Boundary for River Rch & Prof#=Miller Creek,Reach-1,1
Up Type=0
Dn Type=3
Dn Slope=0.005
Boundary for River Rch & Prof#=Miller Creek,Reach-1,2
Up Type=0
Dn Type=3
Dn Slope=0.005
Boundary for River Rch & Prof#=Miller Creek,Reach-1,3
Up Type=0
Dn Type=3
Dn Slope=0.005
Boundary for River Rch & Prof#=Miller Creek,Reach-1,4
Up Type=0
Dn Type=3
Dn Slope=0.005
Boundary for River Rch & Prof#=Miller Creek,Reach-1,5
Up Type=0
Dn Type=3
Dn Slope=0.005
Boundary for River Rch & Prof#=Miller Creek,Reach-1,6
Up Type=0
Dn Type=3
Dn Slope=0.005
Boundary for River Rch & Prof#=Miller Creek,Reach-1,7
Up Type=0
Dn Type=3
Dn Slope=0.005

--- Miller Creek.g01 (geometry) ---

Geom Title=Existing Conditions

River Reach=Miller Creek,Reach-1
Reach XY= 30
      2169487.57     13846375.00      2169241.79     13846708.56
      2168730.42     13847072.33      2168525.07     13847790.39
      2168621.33     13848073.42      2167980.46     13848922.55
      2167919.48     13849277.43      2167266.96     13850331.33
      2166475.00     13850875.00      2166521.89     13851023.37
      2166282.60     13851371.66      2166375.12     13851602.30
      2166224.61     13852202.20      2166573.80     13853214.49
      2165775.07     13854495.03      2165880.52     13855227.43
      2166121.67     13855433.05      2166280.83     13855927.30
      2167132.96     13857381.31      2167321.63     13857476.26
      2167425.23     13858499.93      2167311.63     13859288.32
      2166222.70     13859680.83      2166078.43     13860023.78
      2166684.68     13860335.78      2167276.72     13860921.66
      2167740.21     13860725.51      2168131.07     13860833.13
      2168380.45     13861477.47      2168525.00     13861575.00

Type RM Length L Ch R = 1,20856,344,344,344
BEGIN DESCRIPTION:
Miller Creek 44.0
END DESCRIPTION:
XS GIS Cut Line= 3
      2169113.74     13846073.72      2169476.41     13846408.07
      2169477.27     13846829.29
#Sta/Elev= 30
  4508.0 1210.04  4566.2 1207.17  4602.0 1202.50  4679.6 1199.57  4700.6 1195.58
  4708.0 1193.23  4734.5 1189.48  4799.9 1179.81  4884.9 1162.11  4920.1 1153.29
  4948.4 1143.97  4955.8 1137.43  4962.6 1129.54  4970.0 1124.54  4976.8 1117.85
  4984.2 1113.61  4994.1 1111.88  4994.6 1111.38  4999.7 1111.88  5008.2 1115.48
  5028.2 1116.44  5058.2 1119.58  5085.9 1120.31  5188.2 1121.04  5258.2 1125.43
  5268.2 1128.85  5278.2 1130.15  5318.2 1131.85  5404.3 1131.05  5422.5 1131.41
#Mann=6,-1,0
  4508.0   0.035       0  4734.5    0.12       0  4994.1    0.05       0
  4999.7    0.12       0  5085.9    0.07       0  5404.3   0.035       0
Bank Sta=4994.1,4999.7
Exp/Cntr=0.3,0.1

Type RM Length L Ch R = 1,20512,449,449,449
BEGIN DESCRIPTION:
Miller Creek 43.0
END DESCRIPTION:
XS GIS Cut Line= 3
      2169074.98     13846374.97      2169275.00     13846675.00
      2169325.00     13846825.00
#Sta/Elev= 30
  4638.9 1199.97  4647.7 1199.70  4667.5 1197.97  4688.5 1188.93  4711.0 1181.28
  4724.6 1175.65  4733.6 1170.89  4739.6 1169.24  4754.6 1161.15  4760.6 1159.92
  4769.6 1154.25  4775.6 1153.92  4783.2 1148.21  4805.7 1136.73  4811.7 1135.44
  4826.7 1127.79  4841.7 1123.93  4883.8 1117.06  4898.8 1116.10  4934.9 1115.92
  4940.9 1114.16  4949.9 1113.53  4970.9 1114.79  5007.2 1111.83  5007.7 1111.33
  5012.8 1111.83  5041.7 1118.90  5059.2 1120.60  5115.4 1126.11  5157.6 1127.97
#Mann=5,-1,0
  4638.9   0.035       0  4647.7    0.12       0  5007.2    0.05       0
  5012.8    0.12       0  5059.2    0.07       0
Bank Sta=5007.2,5012.8
Exp/Cntr=0.3,0.1

Type RM Length L Ch R = 1,20063,421,421,421
BEGIN DESCRIPTION:
Miller Creek 42.0
END DESCRIPTION:
XS GIS Cut Line= 3
      2168565.94     13846449.58      2168925.00     13846925.00
      2169150.93     13847162.12
#Sta/Elev= 30
  4404.2 1164.16  4422.4 1162.51  4428.7 1164.04  4443.2 1160.79  4478.6 1161.30
  4493.2 1158.16  4499.4 1159.94  4507.7 1158.12  4514.0 1160.01  4528.6 1159.43
  4543.1 1155.91  4578.5 1158.61  4593.1 1155.45  4607.6 1155.36  4613.9 1157.70
  4649.3 1159.48  4736.7 1158.18  4757.5 1154.16  4813.7 1127.29  4828.3 1122.84
  4857.4 1117.73  4921.9 1113.13  4986.4 1111.69  5004.3 1108.09  5004.7 1107.59
  5009.9 1108.09  5049.5 1115.53  5133.5 1119.31  5233.5 1123.47  5327.5 1123.32
#Mann=4,-1,0
  4404.2    0.12       0  5004.3    0.05       0  5009.9    0.12       0
  5133.5    0.07       0
Bank Sta=5004.3,5009.9
Exp/Cntr=0.3,0.1

Type RM Length L Ch R = 1,19642,486,486,486
BEGIN DESCRIPTION:
Miller Creek 41.0
END DESCRIPTION:
XS GIS Cut Line= 3
      2168524.95     13847225.00      2168675.00     13847225.00
      2169074.95     13847225.00
#Sta/Elev= 30
  4845.3 1130.15  4895.3 1127.06  4905.3 1125.33  4925.3 1115.12  4935.3 1112.18
  4945.3 1110.80  4975.3 1109.53  4985.3 1108.54  4997.8 1108.72  5006.2 1106.05
  5012.3 1103.48  5012.8 1102.98  5017.9 1102.98  5018.4 1103.48  5025.3 1104.32
  5035.3 1106.50  5045.3 1108.06  5055.3 1108.74  5085.3 1109.86  5104.7 1108.43
  5115.3 1108.55  5125.3 1111.91  5135.3 1113.55  5155.3 1112.60  5203.3 1112.75
  5245.3 1114.16  5275.3 1116.54  5355.3 1119.89  5375.3 1122.24  5395.3 1121.88
#Mann=6,-1,0
  4845.3    0.12       0  5006.2   0.035       0  5012.3    0.05       0
  5018.4   0.035       0  5104.7    0.07       0  5203.3   0.035       0
Bank Sta=5012.3,5018.4
Exp/Cntr=0.3,0.1

Type RM Length L Ch R = 1,19156,442,442,442
BEGIN DESCRIPTION:
Miller Creek 40.0
END DESCRIPTION:
XS GIS Cut Line= 3
      2168424.97     13847574.98      2168575.00     13847675.00
      2168974.99     13848024.99
#Sta/Elev= 30
  4814.8 1123.69  4879.4 1117.78  4900.5 1114.15  4915.5 1107.79  4923.0 1103.03
  4966.6 1103.91  4993.5 1101.27  4998.4 1101.27  4999.2 1099.23  4999.7 1098.73
  5005.3 1099.23  5008.9 1099.45  5016.5 1103.83  5030.7 1107.11  5051.6 1105.60
  5104.4 1104.95  5114.8 1105.00  5200.6 1105.14  5249.9 1106.33  5271.8 1108.32
  5292.7 1108.19  5342.0 1109.91  5363.8 1112.10  5392.3 1116.16  5427.4 1119.03
  5455.9 1123.40  5476.8 1125.63  5498.6 1126.87  5503.5 1126.54  5526.6 1127.73
#Mann=7,-1,0
  4814.8    0.12       0  4993.5   0.035       0  4999.2   0.035       0
  5005.3   0.035       0  5104.4    0.12       0  5114.8    0.07       0
  5503.5    0.12       0
Bank Sta=4999.2,5005.3
Exp/Cntr=0.3,0.1

Type RM Length L Ch R = 1,18714,447,447,447
BEGIN DESCRIPTION:
Miller Creek 39.0
END DESCRIPTION:
XS GIS Cut Line= 3
      2168224.97     13847674.97      2168625.00     13848075.00
      2168674.99     13848174.97
#Sta/Elev= 30
  4438.7 1124.49  4452.9 1125.14  4467.0 1124.73  4495.3 1120.91  4537.7 1118.51
  4551.9 1115.74  4615.9 1111.96  4679.2 1109.08  4707.4 1109.18  4721.6 1109.93
  4735.7 1107.23  4848.9 1101.76  4877.2 1101.33  4919.6 1102.18  4962.0 1101.39
  4979.0 1099.95  4990.3 1097.22  5000.9 1095.88  5007.2 1095.88  5015.2 1094.52
  5015.7 1094.02  5021.6 1094.52  5035.2 1094.57  5040.8 1097.51  5049.2 1098.96
  5057.5 1108.28  5063.1 1112.47  5077.7 1114.12  5088.0 1115.01  5116.2 1117.87
#Mann=7,-1,0
  4438.7   0.035       0  4615.9    0.07       0  4979.0    0.12       0
  5015.2    0.05       0  5021.6    0.12       0  5077.7   0.035       0
  5088.0    0.07       0
Bank Sta=5015.2,5021.6
Exp/Cntr=0.3,0.1

Type RM Length L Ch R = 1,18267,446,446,446
BEGIN DESCRIPTION:
Miller Creek 38.0
END DESCRIPTION:
XS GIS Cut Line= 3
      2167890.93     13848146.25      2168375.00     13848425.00
      2168524.99     13848475.00
#Sta/Elev= 30
  4441.4 1121.36  4457.6 1119.67  4493.5 1117.69  4525.1 1118.07  4568.8 1116.57
  4744.9 1108.30  4815.4 1105.95  4847.0 1102.86  4874.3 1101.22  4896.1 1098.64
  4933.2 1098.41  4954.8 1095.65  4970.5 1094.95  4976.9 1095.73  4982.0 1094.01
  4986.3 1092.56  4993.9 1087.04  4994.4 1086.54  5000.4 1087.04  5010.5 1088.10
  5021.1 1092.60  5042.2 1093.47  5063.2 1096.06  5073.8 1099.42  5084.3 1106.13
  5094.9 1111.81  5105.4 1115.37  5137.0 1119.81  5155.5 1124.24  5158.1 1124.24
#Mann=5,-1,0
  4441.4   0.035       0  4568.8    0.07       0  4982.0    0.12       0
  4993.9    0.05       0  5000.4    0.12       0
Bank Sta=4993.9,5000.4
Exp/Cntr=0.3,0.1

Type RM Length L Ch R = 1,17821,478,478,478
BEGIN DESCRIPTION:
Miller Creek 37.0
END DESCRIPTION:
XS GIS Cut Line= 3
      2167889.09     13848577.85      2168125.00     13848775.00
      2168275.04     13848825.01
#Sta/Elev= 30
  4692.3 1110.27  4751.8 1108.04  4857.3 1101.06  4879.4 1100.33  4885.9 1099.30
  4893.7 1099.40  4900.2 1098.45  4908.0 1098.72  4914.5 1097.42  4928.8 1097.51
  4957.4 1095.08  4978.3 1091.75  4986.1 1091.34  4996.5 1088.28  5002.4 1088.28
  5020.8 1084.27  5028.1 1083.91  5028.6 1083.41  5034.2 1083.41  5034.7 1083.91
  5041.9 1084.73  5052.4 1090.75  5063.0 1094.65  5073.5 1099.05  5084.1 1101.28
  5094.6 1102.21  5105.2 1104.32  5115.7 1108.44  5126.2 1111.30  5157.9 1115.75
#Mann=4,-1,0
  4692.3    0.12       0  5028.1    0.05       0  5034.7    0.12       0
  5063.0    0.07       0
Bank Sta=5028.1,5034.7
Exp/Cntr=0.3,0.1

Type RM Length L Ch R = 1,17343,425,425,425
BEGIN DESCRIPTION:
Miller Creek 36.0
END DESCRIPTION:
XS GIS Cut Line= 3
      2167825.01     13849125.00      2167925.00     13849175.00
      2168025.00     13849225.00
#Sta/Elev= 30
  4884.0 1096.19  4898.0 1095.73  4914.7 1094.64  4937.1 1091.06  4942.7 1091.45
  4951.1 1089.15  4959.5 1085.75  4965.0 1085.34  4973.4 1082.15  4981.8 1078.28
  4987.4 1076.23  4993.0 1074.52  4998.6 1074.52  5004.2 1073.78  5006.4 1073.71
  5006.9 1073.21  5012.6 1073.21  5013.1 1073.71  5018.2 1074.89  5026.5 1075.81
  5032.1 1075.23  5040.5 1077.04  5048.9 1082.85  5054.5 1083.38  5056.8 1085.89
  5062.9 1092.53  5071.3 1095.61  5076.9 1095.85  5104.8 1102.16  5107.6 1102.16
#Mann=4,-1,0
  4884.0    0.12       0  5006.4    0.05       0  5013.1    0.12       0
  5056.8    0.07       0
Bank Sta=5006.4,5013.1
Exp/Cntr=0.3,0.1

Type RM Length L Ch R = 1,16918,475,475,475
BEGIN DESCRIPTION:
Miller Creek 35.0
END DESCRIPTION:
XS GIS Cut Line= 3
      2167505.97     13849405.25      2167725.00     13849525.00
      2167991.47     13849688.19
#Sta/Elev= 30
  4750.4 1101.86  4823.1 1099.28  4839.2 1099.59  4866.7 1097.28  4897.5 1096.04
  4904.7 1095.10  4926.5 1089.72  4942.6 1083.87  4948.3 1081.34  4954.4 1077.25
  4964.4 1072.75  4970.1 1071.28  4977.2 1070.51  5003.0 1070.35  5019.8 1068.88
  5020.3 1068.38  5026.6 1068.88  5035.8 1070.84  5058.7 1077.71  5065.8 1081.66
  5071.6 1081.85  5087.1 1087.76  5093.8 1091.67  5117.3 1092.87  5123.8 1093.94
  5181.9 1098.71  5218.6 1101.12  5234.0 1101.63  5239.9 1101.10  5312.5 1107.90
#Mann=4,-1,0
  4750.4    0.12       0  5019.8    0.05       0  5026.6    0.12       0
  5035.8    0.07       0
Bank Sta=5019.8,5026.6
Exp/Cntr=0.3,0.1

Type RM Length L Ch R = 1,16443,450,450,450
BEGIN DESCRIPTION:
Miller Creek 34.0
END DESCRIPTION:
XS GIS Cut Line= 3
      2167037.30     13849689.15      2167525.00     13849925.00
      2168239.96     13850280.06
#Sta/Elev= 30
  4462.2 1112.08  4600.2 1104.60  4782.8 1087.19  4899.5 1077.29  4950.2 1066.15
  4986.1 1063.90  4986.6 1063.40  4993.6 1063.90  5079.6 1067.70  5130.0 1075.63
  5215.2 1077.56  5286.8 1084.96  5365.1 1084.00  5396.0 1084.03  5415.7 1081.45
  5421.2 1087.42  5438.1 1082.43  5443.7 1088.00  5460.5 1080.81  5466.1 1087.15
  5482.9 1084.05  5488.5 1090.12  5505.3 1087.14  5510.9 1091.44  5533.3 1093.54
  5596.3 1086.70  5690.1 1089.62  5712.5 1093.34  5729.4 1108.07  5802.2 1113.62
#Mann=8,-1,0
  4462.2    0.12       0  4782.8    0.07       0  4986.1    0.05       0
  4993.6    0.07       0  5215.2    0.12       0  5365.1   0.035       0
  5396.0    0.12       0  5596.3   0.035       0
Bank Sta=4986.1,4993.6
Exp/Cntr=0.3,0.1

Type RM Length L Ch R = 1,15993,464,464,464
BEGIN DESCRIPTION:
Miller Creek 33.0
END DESCRIPTION:
XS GIS Cut Line= 3
      2167025.03     13850025.03      2167275.00     13850275.00
      2167375.00     13850425.00
#Sta/Elev= 30
  4641.0 1094.15  4669.2 1092.49  4711.7 1085.86  4740.0 1082.92  4747.0 1081.45
  4754.1 1081.01  4782.4 1077.61  4810.7 1073.76  4839.0 1071.06  4858.7 1070.11
  4909.7 1068.81  4923.8 1067.66  4952.1 1061.38  4966.2 1061.23  4980.4 1059.76
  4991.0 1057.79  4998.3 1057.50  4998.8 1057.00  5005.3 1057.00  5005.8 1057.50
  5008.0 1058.47  5017.1 1059.72  5030.6 1060.17  5038.1 1061.94  5044.1 1064.16
  5059.1 1068.13  5095.2 1074.28  5113.6 1076.62  5146.3 1082.10  5174.8 1085.16
#Mann=5,-1,0
  4641.0    0.12       0  4858.7    0.07       0  4998.3    0.05       0
  5005.8    0.07       0  5113.6    0.12       0
Bank Sta=4998.3,5005.8
Exp/Cntr=0.3,0.1

Type RM Length L Ch R = 1,15529,447,447,447
BEGIN DESCRIPTION:
Miller Creek 32.0
END DESCRIPTION:
XS GIS Cut Line= 3
      2166891.52     13850141.28      2166925.00     13850525.00
      2167127.64     13850787.13
#Sta/Elev= 30
  4614.8 1084.39  4713.1 1075.79  4718.9 1074.10  4729.0 1072.76  4759.1 1069.99
  4899.6 1063.31  4919.7 1061.38  4943.6 1058.04  4959.8 1055.06  4969.9 1054.53
  4975.4 1053.58  4979.9 1052.81  4986.1 1050.05  4986.6 1049.55  4993.2 1049.55
  4993.7 1050.05  4997.5 1051.67  5003.1 1051.67  5007.2 1056.36  5021.7 1056.73
  5028.0 1058.08  5042.5 1062.65  5086.0 1067.11  5100.5 1069.25  5135.8 1071.40
  5156.6 1073.44  5220.9 1075.89  5235.4 1075.68  5320.6 1080.43  5331.3 1080.58
#Mann=4,-1,0
  4614.8    0.12       0  4975.4    0.07       0  4986.1    0.05       0
  4993.7    0.07       0
Bank Sta=4986.1,4993.7
Exp/Cntr=0.3,0.1

Type RM Length L Ch R = 1,15082,448,448,448
BEGIN DESCRIPTION:
Miller Creek 31.0
END DESCRIPTION:
XS GIS Cut Line= 3
      2166525.00     13850374.99      2166575.00     13850775.00
      2166975.00     13851175.00
#Sta/Elev= 30
  4596.9 1076.10  4617.1 1075.48  4634.7 1073.61  4657.4 1072.24  4687.6 1068.48
  4720.4 1066.51  4758.2 1062.29  4838.8 1058.57  4889.2 1057.93  4919.4 1053.39
  4939.6 1053.50  4949.6 1052.42  4983.0 1051.57  4989.9 1050.59  4993.7 1049.21
  4994.2 1048.71  5000.8 1048.71  5001.3 1049.21  5014.2 1050.10  5042.4 1057.09
  5069.0 1058.93  5099.0 1061.27  5155.6 1062.72  5226.3 1062.35  5315.0 1063.09
  5339.4 1064.02  5381.9 1067.04  5452.6 1076.87  5495.0 1081.40  5565.7 1090.47
#Mann=6,-1,0
  4596.9   0.035       0  4983.0    0.12       0  4993.7    0.05       0
  5001.3    0.12       0  5069.0    0.07       0  5315.0    0.12       0
Bank Sta=4993.7,5001.3
Exp/Cntr=0.3,0.1

Type RM Length L Ch R = 1,14634,361,361,361
BEGIN DESCRIPTION:
Miller Creek 30.0
END DESCRIPTION:
XS GIS Cut Line= 3
      2164509.41     13851569.65      2166425.00     13851125.00
      2167130.72     13851341.14
#Sta/Elev= 30
  3034.1 1134.97  3081.4 1128.77  3347.8 1115.49  3651.2 1109.79  3736.5 1106.75
  3741.6 1103.78  3784.3 1106.27  3789.4 1103.98  3853.9 1104.44  3943.2 1097.35
  3953.5 1102.06  3965.1 1094.03  4088.5 1084.18  4370.1 1069.75  4487.1 1061.66
  4666.7 1058.23  4774.8 1056.98  4840.5 1052.25  4918.5 1052.29  4954.4 1048.15
  4954.9 1047.65  4964.8 1048.15  5000.1 1051.22  5042.5 1053.28  5087.8 1048.20
  5153.3 1059.08  5377.1 1061.76  5393.1 1067.34  5491.4 1084.34  5738.7 1114.22
#Mann=9,-1,0
  3034.1    0.12       0  3853.9   0.035       0  4088.5    0.07       0
  4370.1    0.12       0  4666.7    0.07       0  4840.5   0.035       0
  4954.4   0.035       0  4964.8   0.035       0  5000.1    0.12       0
Bank Sta=4954.4,4964.8
Exp/Cntr=0.3,0.1

Type RM Length L Ch R = 1,14273,200,200,200
BEGIN DESCRIPTION:
Miller Creek 29.5
END DESCRIPTION:
XS GIS Cut Line= 4
      2165453.89     13851519.86      2166149.25     13851400.07
      2166297.44     13851398.31      2167060.31     13851353.21
#Sta/Elev= 30
  4146.2 1115.11  4299.5 1109.52  4318.4 1105.02  4330.0 1098.00  4378.3 1085.85
  4461.9 1074.44  4498.1 1064.93  4522.8 1062.31  4672.7 1056.68  4786.6 1056.63
  4851.8 1055.72  4877.6 1053.88  4896.9 1055.62  4990.9 1050.92  4991.4 1050.42
  5001.7 1050.92  5077.7 1055.77  5136.8 1052.91  5141.8 1054.01  5158.5 1051.98
  5187.9 1051.78  5238.0 1056.20  5306.7 1058.77  5418.3 1058.64  5481.6 1060.75
  5488.4 1064.48  5508.4 1070.95  5538.5 1076.28  5668.7 1094.44  5764.2 1105.35
#Mann=5,-1,0
  4146.2    0.12       0  4896.9   0.035       0  4990.9   0.035       0
  5001.7   0.035       0  5158.5    0.12       0
Bank Sta=4990.9,5001.7
Exp/Cntr=0.3,0.1

Type RM Length L Ch R = 1,14073,338,338,338
BEGIN DESCRIPTION:
Miller Creek 29.0
END DESCRIPTION:
XS GIS Cut Line= 2
      2165377.05     13851765.68      2167124.12     13851419.66
#Sta/Elev= 30
  3982.2 1137.54  4013.1 1137.34  4082.7 1134.14  4202.7 1118.49  4269.7 1111.64
  4315.8 1093.85  4320.9 1094.57  4357.3 1084.38  4398.1 1077.05  4459.2 1071.01
  4500.0 1060.09  4525.8 1056.92  4594.9 1054.89  4693.7 1052.95  4744.7 1054.93
  4797.0 1051.54  4809.0 1051.14  4910.0 1047.60  4935.6 1045.09  4968.9 1044.76
  4979.1 1046.80  5004.3 1042.57  5004.8 1042.07  5015.2 1042.57  5030.1 1046.21
  5112.1 1054.53  5417.5 1060.55  5458.3 1072.37  5509.2 1080.65  5763.2 1114.41
#Mann=11,-1,0
  3982.2    0.07       0  4013.1    0.12       0  4082.7    0.07       0
  4202.7    0.12       0  4594.9   0.035       0  4797.0    0.12       0
  4809.0   0.035       0  4910.0    0.07       0  5004.3    0.05       0
  5015.2    0.07       0  5112.1    0.12       0
Bank Sta=5004.3,5015.2
Exp/Cntr=0.3,0.1

Type RM Length L Ch R = 1,13735,483,483,483
BEGIN DESCRIPTION:
Miller Creek 28.0
END DESCRIPTION:
XS GIS Cut Line= 3
      2166025.02     13851875.00      2166275.00     13851875.00
      2167074.99     13851775.00
#Sta/Elev= 30
  4745.1 1057.77  4795.1 1056.23  4835.1 1053.78  4855.1 1050.25  4925.1 1045.27
  4985.1 1043.85  4998.5 1042.61  4999.7 1042.21  5000.2 1041.71  5010.6 1042.21
  5015.2 1043.52  5032.9 1044.23  5055.6 1043.35  5085.8 1049.49  5113.5 1050.96
  5237.0 1052.46  5297.4 1054.07  5441.0 1054.29  5509.1 1055.97  5521.7 1057.58
  5529.2 1059.72  5559.4 1071.39  5597.2 1082.21  5602.3 1081.93  5630.0 1088.28
  5660.2 1093.37  5720.7 1101.85  5758.5 1108.19  5763.5 1107.96  5801.3 1112.92
#Mann=4,-1,0
  4745.1   0.035       0  4998.5    0.12       0  4999.7    0.05       0
  5010.6    0.12       0
Bank Sta=4999.7,5010.6
Exp/Cntr=0.3,0.1

Type RM Length L Ch R = 1,13252,463,463,463
BEGIN DESCRIPTION:
Miller Creek 27.0
END DESCRIPTION:
XS GIS Cut Line= 3
      2165769.96     13852245.45      2166275.00     13852325.00
      2167030.20     13852165.64
#Sta/Elev= 30
  4484.1 1066.94  4497.7 1066.08  4570.4 1061.64  4638.9 1058.21  4749.1 1054.35
  4885.8 1050.26  4944.8 1048.54  4985.2 1046.04  4992.8 1039.66  4997.9 1039.66
  5005.6 1034.26  5009.6 1032.74  5010.1 1032.24  5020.6 1032.74  5026.0 1038.10
  5056.7 1040.73  5086.2 1045.07  5164.4 1046.39  5196.5 1048.36  5281.5 1050.64
  5485.9 1051.27  5588.1 1054.28  5602.1 1055.84  5646.8 1063.86  5651.9 1065.82
  5690.3 1074.52  5696.5 1077.15  5746.3 1084.51  5751.7 1086.67  5767.2 1090.05
#Mann=9,-1,0
  4484.1    0.07       0  4497.7    0.12       0  4570.4    0.07       0
  4749.1   0.035       0  4885.8    0.12       0  5009.6    0.05       0
  5020.6    0.12       0  5086.2    0.07       0  5196.5    0.12       0
Bank Sta=5009.6,5020.6
Exp/Cntr=0.3,0.1

Type RM Length L Ch R = 1,12789,455,455,455
BEGIN DESCRIPTION:
Miller Creek 26.0
END DESCRIPTION:
XS GIS Cut Line= 3
      2165599.73     13852691.73      2166475.00     13852725.00
      2167381.80     13852738.58
#Sta/Elev= 30
  4124.1 1064.65  4186.7 1060.63  4375.7 1053.89  4479.4 1050.52  4580.7 1046.68
  4692.3 1044.55  4759.8 1043.75  4876.2 1044.87  4919.9 1043.60  4950.0 1036.95
  4992.0 1033.00  4992.5 1032.50  5003.0 1033.00  5010.0 1035.97  5040.0 1042.32
  5060.0 1043.76  5130.0 1041.00  5160.0 1041.12  5334.5 1047.96  5370.0 1050.49
  5380.0 1052.03  5410.0 1060.33  5440.1 1070.69  5460.1 1080.13  5470.1 1081.83
  5590.1 1093.53  5710.1 1102.58  5740.1 1103.65  5861.2 1114.90  5906.9 1118.69
#Mann=10,-1,0
  4124.1   0.035       0  4186.7    0.07       0  4375.7    0.12       0
  4479.4   0.035       0  4580.7    0.07       0  4692.3   0.035       0
  4876.2    0.12       0  4992.0    0.05       0  5003.0    0.12       0
  5861.2    0.07       0
Bank Sta=4992,5003
Exp/Cntr=0.3,0.1

Type RM Length L Ch R = 1,12334,382,382,382
BEGIN DESCRIPTION:
Miller Creek 25.0
END DESCRIPTION:
XS GIS Cut Line= 3
      2165464.30     13852915.68      2166575.00     13853125.00
      2167065.93     13853129.23
#Sta/Elev= 30
  3869.3 1073.86  3900.5 1068.47  3946.5 1062.87  3963.2 1063.85  3981.9 1063.54
  4046.8 1057.18  4124.4 1051.94  4301.9 1045.21  4460.2 1041.51  4663.7 1040.47
  4805.8 1041.29  4860.4 1039.75  4887.6 1040.29  4920.9 1038.81  4968.2 1032.91
  4989.4 1032.11  4991.4 1030.32  4991.9 1029.82  5002.7 1030.32  5039.5 1034.16
  5059.5 1040.23  5099.6 1043.26  5129.6 1048.00  5179.6 1069.92  5189.6 1080.44
  5199.6 1084.68  5259.6 1092.96  5299.6 1096.80  5399.6 1103.79  5490.5 1108.05
#Mann=7,-1,0
  3869.3   0.035       0  3963.2    0.07       0  4046.8    0.12       0
  4301.9   0.035       0  4860.4    0.12       0  4991.4    0.05       0
  5002.7    0.12       0
Bank Sta=4991.4,5002.7
Exp/Cntr=0.3,0.1

Type RM Length L Ch R = 1,11952,563,563,563
BEGIN DESCRIPTION:
Miller Creek 24.0
END DESCRIPTION:
XS GIS Cut Line= 2
      2165195.74     13852851.84      2166833.77     13853649.44
#Sta/Elev= 30
  3614.3 1117.03  3676.6 1114.40  3688.5 1110.65  3704.7 1103.00  3744.3 1092.15
  3865.8 1078.13  3904.5 1070.42  3947.2 1064.42  4025.9 1062.06  4079.2 1055.41
  4228.4 1047.54  4336.4 1043.04  4552.4 1039.23  4584.8 1039.09  4824.5 1036.85
  4888.1 1037.30  4916.2 1036.08  4948.2 1031.55  4983.9 1033.28  5023.3 1027.81
  5023.8 1027.31  5034.6 1027.81  5037.2 1031.49  5051.5 1040.69  5091.0 1050.89
  5209.3 1064.20  5248.5 1072.83  5260.0 1076.85  5276.9 1086.24  5436.2 1108.46
#Mann=12,-1,0
  3614.3    0.12       0  3688.5    0.07       0  3865.8   0.035       0
  3904.5    0.07       0  4079.2    0.12       0  4228.4    0.07       0
  4336.4   0.035       0  4552.4    0.07       0  4584.8   0.035       0
  4824.5    0.12       0  5023.3    0.05       0  5034.6    0.12       0
Bank Sta=5023.3,5034.6
Exp/Cntr=0.3,0.1

Type RM Length L Ch R = 1,11389,470,470,470
BEGIN DESCRIPTION:
Miller Creek 23.0
END DESCRIPTION:
XS GIS Cut Line= 3
      2165675.01     13853775.00      2166075.00     13853875.00
      2166474.99     13854075.00
#Sta/Elev= 30
  4583.4 1044.02  4614.3 1041.75  4637.6 1038.94  4655.5 1037.86  4676.2 1039.88
  4779.2 1036.89  4854.0 1035.84  4913.2 1033.63  4945.8 1030.47  4977.7 1027.56
  4985.4 1028.53  4998.5 1027.85  5003.8 1026.34  5004.3 1025.84  5015.5 1026.34
  5018.1 1027.31  5032.0 1027.18  5054.4 1029.61  5076.8 1030.09  5107.5 1035.10
  5138.2 1033.74  5166.2 1034.79  5183.0 1036.71  5188.6 1035.83  5196.9 1036.03
  5250.0 1041.41  5308.7 1044.29  5353.5 1048.23  5406.6 1056.77  5442.9 1061.03
#Mann=5,-1,0
  4583.4    0.12       0  4637.6   0.035       0  4945.8    0.12       0
  5003.8    0.05       0  5015.5    0.12       0
Bank Sta=5003.8,5015.5
Exp/Cntr=0.3,0.1

Type RM Length L Ch R = 1,10919,434,434,434
BEGIN DESCRIPTION:
Miller Creek 22.0
END DESCRIPTION:
XS GIS Cut Line= 3
      2165525.01     13854275.00      2165875.00     13854275.00
      2166275.00     13854325.00
#Sta/Elev= 30
  4650.4 1052.13  4670.4 1051.74  4710.4 1042.59  4730.4 1040.19  4739.7 1039.57
  4790.4 1037.98  4810.4 1036.54  4820.4 1034.86  4830.4 1031.00  4840.4 1027.99
  4850.4 1027.41  4900.4 1027.75  4960.4 1025.32  4980.4 1025.81  4990.4 1025.34
  4997.9 1024.28  5037.4 1023.93  5037.9 1023.43  5048.6 1023.43  5049.1 1023.93
  5062.0 1025.93  5081.0 1026.13  5118.8 1029.22  5161.6 1030.85  5252.3 1032.20
  5272.5 1033.47  5285.1 1033.16  5292.6 1034.06  5322.9 1035.15  5403.5 1042.00
#Mann=5,-1,0
  4650.4    0.12       0  4739.7   0.035       0  5037.4   0.035       0
  5049.1   0.035       0  5062.0    0.12       0
Bank Sta=5037.4,5049.1
Exp/Cntr=0.3,0.1

Type RM Length L Ch R = 1,10485,482,482,482
BEGIN DESCRIPTION:
Miller Creek 21.0
END DESCRIPTION:
XS GIS Cut Line= 3
      2165249.20     13854703.79      2165775.00     13854675.00
      2166299.97     13854492.43
#Sta/Elev= 30
  4473.5 1074.21  4489.3 1074.61  4519.4 1071.13  4590.1 1065.77  4649.6 1058.03
  4727.8 1052.00  4739.7 1051.81  4759.7 1047.00  4799.8 1041.73  4889.9 1036.82
  4906.8 1032.76  4960.0 1027.01  4990.1 1020.75  4997.6 1016.17  5004.4 1016.16
  5004.9 1015.66  5016.2 1016.16  5021.3 1019.73  5044.9 1022.83  5053.0 1023.23
  5063.6 1019.78  5077.8 1018.08  5095.4 1022.07  5103.7 1025.56  5116.5 1026.98
  5253.9 1027.98  5455.3 1032.66  5518.9 1037.17  5533.8 1039.43  5555.9 1044.96
#Mann=6,-1,0
  4473.5   0.035       0  4590.1    0.12       0  4727.8   0.035       0
  5004.4   0.035       0  5016.2   0.035       0  5044.9    0.12       0
Bank Sta=5004.4,5016.2
Exp/Cntr=0.3,0.1

Type RM Length L Ch R = 1,10003,424,424,424
BEGIN DESCRIPTION:
Miller Creek 20.0
END DESCRIPTION:
XS GIS Cut Line= 3
      2165183.16     13855158.65      2165875.00     13855125.00
      2166274.97     13854725.03
#Sta/Elev= 30
  4311.9 1089.00  4322.1 1087.58  4333.8 1084.82  4353.8 1086.16  4373.8 1084.98
  4413.9 1080.04  4473.9 1070.49  4524.0 1066.67  4589.4 1055.42  4624.1 1052.25
  4664.2 1042.85  4692.5 1039.56  4717.2 1038.49  4784.3 1032.36  4884.4 1029.25
  4954.5 1024.78  4964.5 1022.87  4978.6 1013.84  4979.1 1013.34  4990.4 1013.84
  5008.1 1014.62  5018.7 1016.89  5131.8 1023.17  5216.7 1024.51  5329.8 1023.52
  5414.7 1026.63  5457.1 1029.62  5513.7 1031.58  5556.1 1037.00  5570.2 1037.25
#Mann=6,-1,0
  4311.9   0.035       0  4322.1    0.07       0  4589.4   0.035       0
  4717.2    0.12       0  4978.6    0.05       0  4990.4    0.12       0
Bank Sta=4978.6,4990.4
Exp/Cntr=0.3,0.1

Type RM Length L Ch R = 1,9579,460,460,460
BEGIN DESCRIPTION:
Miller Creek 19.0
END DESCRIPTION:
XS GIS Cut Line= 3
      2165724.98     13855825.02      2166125.00     13855425.00
      2166525.00     13855025.00
#Sta/Elev= 30
  4441.9 1061.70  4526.8 1053.60  4555.1 1046.05  4569.2 1043.56  4639.9 1038.19
  4654.1 1034.88  4710.6 1032.42  4823.8 1024.68  4837.9 1021.67  4852.1 1016.56
  4866.2 1014.14  4894.5 1014.55  4908.6 1016.37  4922.8 1015.16  4936.9 1016.06
  4951.0 1014.66  4973.4 1010.09  4973.9 1009.59  4985.3 1010.09  4993.5 1016.63
  5004.1 1019.15  5035.9 1020.44  5191.5 1019.23  5233.9 1021.03  5375.3 1030.61
  5446.0 1033.83  5488.4 1039.52  5530.9 1041.76  5569.8 1051.00  5573.3 1051.00
#Mann=3,-1,0
  4441.9    0.12       0  4973.4    0.05       0  4985.3    0.12       0
Bank Sta=4973.4,4985.3
Exp/Cntr=0.3,0.1

Type RM Length L Ch R = 1,9119,441,441,441
BEGIN DESCRIPTION:
Miller Creek 18.0
END DESCRIPTION:
XS GIS Cut Line= 3
      2165875.00     13856025.00      2166225.00     13855825.00
      2166624.98     13855725.01
#Sta/Elev= 30
  4593.0 1065.54  4681.5 1054.34  4708.9 1045.95  4731.2 1042.71  4762.2 1039.76
  4799.6 1034.05  4834.9 1032.02  4880.2 1025.74  4915.5 1022.88  4938.5 1019.71
  4960.8 1014.74  4988.2 1012.88  4993.2 1010.68  4998.7 1010.68  5000.5 1009.05
  5001.0 1008.55  5012.4 1009.05  5027.0 1011.37  5037.3 1011.93  5068.3 1010.09
  5088.9 1011.40  5109.5 1015.47  5130.1 1016.97  5171.3 1016.80  5274.4 1014.33
  5295.0 1015.92  5315.7 1019.51  5356.9 1030.35  5367.2 1031.34  5408.4 1031.92
#Mann=3,-1,0
  4593.0    0.12       0  5000.5    0.05       0  5012.4    0.12       0
Bank Sta=5000.5,5012.4
Exp/Cntr=0.3,0.1

Type RM Length L Ch R = 1,8678,409,409,409
BEGIN DESCRIPTION:
Miller Creek 17.0
END DESCRIPTION:
XS GIS Cut Line= 3
      2166125.03     13856374.98      2166475.00     13856175.00
      2166875.02     13855924.99
#Sta/Elev= 30
  4601.5 1065.53  4624.5 1062.97  4674.2 1053.76  4711.6 1043.36  4770.6 1034.18
  4808.1 1030.97  4820.3 1026.24  4866.4 1017.26  4916.0 1013.01  4931.9 1009.61
  4959.2 1007.03  4975.6 1003.85  4976.1 1003.35  4987.5 1003.85  4996.7 1005.40
  5001.7 1007.96  5033.5 1010.12  5048.8 1013.15  5098.9 1014.05  5193.3 1012.13
  5222.1 1015.96  5252.2 1022.49  5264.6 1026.87  5295.3 1031.80  5346.6 1034.39
  5381.9 1039.63  5410.8 1040.47  5432.1 1044.24  5447.4 1050.37  5476.3 1051.99
#Mann=3,-1,0
  4601.5    0.12       0  4975.6    0.05       0  4987.5    0.12       0
Bank Sta=4975.6,4987.5
Exp/Cntr=0.3,0.1

Type RM Length L Ch R = 1,8269,440,440,440
BEGIN DESCRIPTION:
Miller Creek 16.0
END DESCRIPTION:
XS GIS Cut Line= 3
      2166474.97     13856625.02      2166625.00     13856525.00
      2167024.99     13856225.01
#Sta/Elev= 30
  4815.2 1033.22  4843.8 1031.45  4864.8 1024.60  4894.9 1018.26  4930.9 1013.81
  4936.9 1012.56  4945.9 1007.41  4959.5 1003.71  4967.0 1005.48  4998.6 1005.76
  5003.1 1002.08  5003.6 1001.58  5015.0 1002.08  5023.6 1005.06  5045.5 1006.85
  5067.4 1011.24  5088.2 1011.57  5167.4 1008.88  5209.1 1009.01  5223.6 1011.15
  5259.1 1019.17  5288.2 1028.78  5302.8 1032.00  5338.2 1032.82  5367.4 1036.75
  5423.6 1039.60  5434.9 1041.10  5455.5 1045.24  5482.0 1050.99  5495.5 1051.75
#Mann=5,-1,0
  4815.2    0.12       0  5003.1    0.05       0  5015.0    0.12       0
  5434.9    0.07       0  5455.5    0.12       0
Bank Sta=5003.1,5015
Exp/Cntr=0.3,0.1

Type RM Length L Ch R = 1,7829,469,469,469
BEGIN DESCRIPTION:
Miller Creek 15.0
END DESCRIPTION:
XS GIS Cut Line= 3
      2166474.98     13856875.00      2166875.00     13856875.00
      2167074.98     13856775.01
#Sta/Elev= 30
  4604.6 1042.01  4624.6 1040.77  4644.6 1037.00  4664.6 1034.27  4714.6 1031.44
  4724.6 1030.11  4754.6 1021.62  4774.6 1017.42  4794.6 1014.48  4834.6 1010.57
  4864.6 1005.80  4885.2 1005.16  4924.6 1004.14  4944.6 1001.61  4978.6 1000.99
  4979.1 1000.49  4990.7 1000.99  4994.6 1001.15  5002.1 1003.34  5004.9 1003.34
  5018.6 1002.80  5063.3 1005.91  5138.8 1005.70  5152.8 1008.14  5161.1 1012.43
  5175.1 1016.91  5191.9 1024.39  5205.9 1028.69  5214.2 1030.65  5228.2 1030.95
#Mann=5,-1,0
  4604.6    0.12       0  4885.2   0.035       0  4978.6   0.035       0
  4990.7   0.035       0  5004.9    0.12       0
Bank Sta=4978.6,4990.7
Exp/Cntr=0.3,0.1

Type RM Length L Ch R = 1,7360,455,455,455
BEGIN DESCRIPTION:
Miller Creek 14.0
END DESCRIPTION:
XS GIS Cut Line= 3
      2166675.04     13857524.98      2167075.00     13857275.00
      2167225.02     13856974.97
#Sta/Elev= 30
  4522.0 1054.72  4550.8 1051.12  4566.2 1045.71  4587.4 1042.50  4624.0 1040.12
  4660.5 1034.39  4703.0 1032.07  4754.9 1018.92  4791.4 1013.65  4797.3 1016.17
  4805.0 1015.15  4812.6 1013.92  4818.5 1009.93  4840.3 1006.89  4904.9 1004.94
  4958.3 1005.32  4970.7 1000.37  4974.0  995.56  4974.5  995.06  4986.2  995.56
  4990.7  997.03  5024.4  996.89  5052.3 1001.08  5060.7 1000.29  5097.1 1003.11
  5150.2 1002.11  5208.9 1003.18  5231.2 1007.04  5292.7 1028.19  5329.1 1030.39
#Mann=4,-1,0
  4522.0   0.035       0  4904.9    0.12       0  4974.0    0.05       0
  4986.2    0.12       0
Bank Sta=4974,4986.2
Exp/Cntr=0.3,0.1

Type RM Length L Ch R = 1,6905,458,458,458
BEGIN DESCRIPTION:
Miller Creek 13.0
END DESCRIPTION:
XS GIS Cut Line= 3
      2167025.01     13857725.00      2167325.00     13857575.00
      2168425.02     13857975.01
#Sta/Elev= 30
  4664.5 1032.48  4700.8 1030.55  4731.6 1019.43  4798.7 1000.87  4821.0  999.25
  4859.3 1000.11  4946.8  996.84  4975.7  993.83  4982.8  992.86  4983.3  992.36
  5000.2  992.86  5009.9  995.98  5015.2  995.56  5021.2  998.73  5046.2 1001.63
  5169.0 1002.81  5483.4 1003.14  5595.1 1005.61  5656.3 1011.42  5686.9 1010.98
  5734.1 1014.19  5795.1 1022.88  5821.3 1026.02  5834.5 1028.26  5890.4 1030.11
  6004.3 1040.47  6038.0 1047.09  6099.2 1054.48  6124.5 1060.04  6170.4 1062.33
#Mann=10,-1,0
  4664.5    0.12       0  4859.3    0.07       0  4975.7    0.12       0
  4982.8    0.05       0  5000.2    0.12       0  5046.2    0.07       0
  5169.0   0.035       0  5795.1    0.07       0  5821.3   0.035       0
  6004.3    0.12       0
Bank Sta=4982.8,5000.2
Exp/Cntr=0.3,0.1

Type RM Length L Ch R = 1,6447,380,380,380
BEGIN DESCRIPTION:
Miller Creek 12.0
END DESCRIPTION:
XS GIS Cut Line= 3
      2167125.01     13857875.01      2167375.00     13858025.00
      2167874.96     13858124.99
#Sta/Elev= 30
  4718.9 1025.81  4742.2 1025.47  4753.9 1023.67  4785.0 1014.23  4800.5 1011.95
  4821.9 1005.51  4827.7 1005.57  4838.3 1001.52  4843.3  999.23  4849.1  999.34
  4858.8  995.39  4870.5  993.46  4944.4  993.91  4965.7  993.39  4978.4  991.65
  4978.9  991.15  4995.9  991.65  5007.5  994.74  5013.0  994.74  5020.6  997.38
  5030.8  998.98  5112.4  998.33  5336.8 1000.12  5367.4 1003.24  5387.8 1007.85
  5418.4 1009.41  5428.6 1013.31  5469.3 1024.97  5489.7 1028.49  5520.3 1030.02
#Mann=5,-1,0
  4718.9    0.12       0  4838.3    0.07       0  4978.4    0.05       0
  4995.9    0.07       0  5013.0   0.035       0
Bank Sta=4978.4,4995.9
Exp/Cntr=0.3,0.1

Type RM Length L Ch R = 1,6067,539,539,539
BEGIN DESCRIPTION:
Miller Creek 11.0
END DESCRIPTION:
XS GIS Cut Line= 3
      2166775.02     13857875.02      2167367.22     13858366.98
      2168040.39     13858516.19
#Sta/Elev= 30
  4222.5 1054.72  4250.5 1052.39  4307.8 1042.15  4371.6 1039.26  4421.0 1032.76
  4486.1 1028.85  4563.0 1016.24  4614.1 1011.68  4618.9 1011.31  4684.1 1003.97
  4783.0  998.99  4805.2  998.19  4811.7 1000.87  4826.0 1001.41  4869.0 1000.92
  4883.3  998.73  4889.8  994.77  4897.6  993.74  4991.6  988.97  4992.1  988.47
  5009.2  988.97  5011.8  990.94  5049.5  999.08  5154.0  996.15  5266.7  996.45
  5317.9 1007.79  5384.2 1026.59  5410.1 1030.15  5588.7 1040.12  5681.9 1047.52
#Mann=9,-1,0
  4222.5   0.035       0  4486.1    0.12       0  4614.1    0.07       0
  4618.9   0.035       0  4991.6   0.035       0  5009.2   0.035       0
  5011.8    0.12       0  5384.2   0.035       0  5588.7    0.12       0
Bank Sta=4991.6,5009.2
Exp/Cntr=0.3,0.1

Type RM Length L Ch R = 1,5528,484,484,484
BEGIN DESCRIPTION:
Miller Creek 10.0
END DESCRIPTION:
XS GIS Cut Line= 3
      2166775.02     13858275.02      2167375.00     13858875.00
      2167575.00     13858875.00
#Sta/Elev= 30
  4151.5 1030.67  4179.8 1027.34  4222.2 1016.92  4264.6 1010.98  4292.9 1005.84
  4335.3 1003.05  4349.5 1001.19  4476.7  996.77  4660.6  997.84  4874.6  996.81
  4901.0  996.97  4943.4  994.95  4957.6  993.40  4996.5  983.69  5000.0  983.69
  5001.1  981.23  5001.6  980.73  5018.8  981.23  5020.0  982.47  5030.0  986.48
  5060.0  989.39  5090.0  987.96  5110.0  991.20  5120.0  994.80  5130.0 1000.36
  5150.0 1014.49  5160.0 1019.51  5170.0 1022.97  5180.0 1024.50  5200.0 1025.23
#Mann=4,-1,0
  4151.5   0.035       0  4874.6    0.12       0  5001.1    0.05       0
  5018.8    0.12       0
Bank Sta=5001.1,5018.8
Exp/Cntr=0.3,0.1

Type RM Length L Ch R = 1,5044,456,456,456
BEGIN DESCRIPTION:
Miller Creek 9.0
END DESCRIPTION:
XS GIS Cut Line= 3
      2166374.99     13858324.99      2167275.00     13859325.00
      2167474.97     13859275.01
#Sta/Elev= 30
  3654.1 1062.92  3788.6 1051.42  3816.7 1042.96  3830.9 1040.35  3866.8 1038.07
  3909.4 1031.16  3951.2 1028.98  3965.4 1026.26  4008.0 1013.32  4064.8 1002.19
  4093.2 1002.26  4121.6  997.02  4188.3  994.91  4301.5  993.80  4849.4  993.55
  4907.2  993.79  4935.6  991.00  4978.2  980.77  5000.9  976.82  5001.4  976.32
  5018.6  976.82  5030.4  978.58  5040.7  978.01  5051.0  980.07  5058.7  984.55
  5063.9  980.83  5100.0  999.83  5164.4 1000.34  5187.6 1001.38  5205.6 1003.88
#Mann=6,-1,0
  3654.1   0.035       0  4188.3    0.07       0  4301.5   0.035       0
  4849.4    0.12       0  5000.9    0.05       0  5018.6    0.12       0
Bank Sta=5000.9,5018.6
Exp/Cntr=0.3,0.1

Type RM Length L Ch R = 1,4588,515,515,515
BEGIN DESCRIPTION:
Miller Creek 8.0
END DESCRIPTION:
XS GIS Cut Line= 4
      2166275.00     13858875.00      2166875.00     13859475.00
      2167054.91     13859523.17      2167649.50     13859317.61
#Sta/Elev= 30
  4151.4 1014.91  4154.9 1014.91  4186.8 1003.35  4222.1 1001.84  4264.5  993.22
  4285.5  991.89  4314.0  991.28  4781.9  990.65  4858.5  990.82  4886.8  991.94
  4957.5  984.59  4971.6  981.62  4987.5  975.39  4988.0  974.89  5005.2  975.39
  5057.4  977.30  5062.6  981.74  5082.7  983.27  5092.3  985.81  5097.4  996.68
  5103.5  997.08  5113.8  995.42  5132.3  998.38  5137.5 1000.30  5318.4 1000.62
  5593.7  998.01  5599.0  998.89  5768.2 1002.52  5789.4 1004.77  5815.3 1005.74
#Mann=6,-1,0
  4151.4   0.035       0  4285.5    0.07       0  4314.0   0.035       0
  4781.9    0.12       0  4987.5    0.05       0  5005.2    0.12       0
Bank Sta=4987.5,5005.2
Exp/Cntr=0.3,0.1

Type RM Length L Ch R = 1,4073,478,478,478
BEGIN DESCRIPTION:
Miller Creek 7.2
END DESCRIPTION:
XS GIS Cut Line= 4
      2165686.76     13859209.80      2166587.91     13859696.39
      2167093.55     13859610.01      2167744.80     13859335.33
#Sta/Elev= 30
  4185.7 1021.31  4269.6 1019.94  4285.8 1017.57  4307.7 1013.64  4329.6 1004.29
  4365.5 1002.44  4379.1  994.24  4400.9  989.42  4487.9  987.82  4532.1  987.91
  4814.6  987.61  4837.9  987.92  4865.6  981.66  4970.8  978.78  4985.4  977.90
  4992.8  974.89  4993.3  974.39  5010.5  974.89  5013.3  977.45  5038.7  979.30
  5067.3  984.01  5073.0  987.43  5104.2  989.17  5359.0  988.83  5453.5  991.88
  5612.7  996.39  5956.1  996.97  6080.1  994.06  6321.3 1002.60  6429.6 1011.42
#Mann=9,-1,0
  4185.7   0.035       0  4487.9    0.07       0  4532.1   0.035       0
  4814.6    0.12       0  4970.8    0.07       0  4992.8    0.05       0
  5010.5    0.07       0  5038.7   0.035       0  5453.5    0.12       0
Bank Sta=4992.8,5010.5
Exp/Cntr=0.3,0.1

Type RM Length L Ch R = 1,3595,328,328,328
BEGIN DESCRIPTION:
Miller Creek 7.1
END DESCRIPTION:
XS GIS Cut Line= 4
      2165154.55     13860035.33      2166073.94     13859891.80
      2166858.88     13859765.05      2167860.90     13859327.56
#Sta/Elev= 30
  4068.7 1016.34  4234.5 1013.50  4336.7 1008.78  4427.9 1005.04  4458.4 1000.87
  4501.1  995.85  4558.6  988.55  4631.8  986.37  4746.9  985.03  4959.4  988.17
  4969.9  986.02  4999.0  973.32  4999.5  972.82  5016.8  973.32  5030.7  976.68
  5074.8  976.54  5120.8  979.46  5156.6  980.56  5172.5  983.83  5203.3  984.15
  5223.1  988.44  5260.3  988.34  5830.1  987.40  5954.8  992.91  6132.8  995.07
  6430.1  992.92  6581.4  997.27  6703.9 1003.88  6794.0 1011.61  6887.7 1024.48
#Mann=12,-1,0
  4068.7    0.07       0  4336.7    0.12       0  4458.4    0.07       0
  4501.1    0.12       0  4631.8   0.035       0  4959.4    0.07       0
  4999.0    0.05       0  5016.8    0.07       0  5120.8   0.035       0
  5156.6    0.07       0  5260.3   0.035       0  5954.8    0.12       0
Bank Sta=4999,5016.8
Exp/Cntr=0.3,0.1

Type RM Length L Ch R = 1,3267,501,501,501
BEGIN DESCRIPTION:
Miller Creek 7.0
END DESCRIPTION:
XS GIS Cut Line= 3
      2165816.91     13860409.04      2166350.36     13860021.45
      2167857.36     13859366.13
#Sta/Elev= 30
  4468.7  994.24  4575.8  992.32  4599.7  991.80  4857.0  987.77  4886.4  985.08
  4913.5  980.17  4942.8  979.73  4957.5  977.23  4963.7  974.45  4969.4  969.79
  4969.9  969.29  4987.3  969.79  5013.9  971.92  5022.8  974.15  5028.6  977.52
  5058.0  979.41  5097.9  985.88  5121.5  987.79  5235.7  988.15  5782.8  986.72
  5829.7  987.60  5858.6  989.32  5864.1  990.90  5899.0  991.52  6062.5  994.09
  6284.4  991.87  6376.3  992.96  6605.3 1002.77  6703.4 1011.73  6771.4 1020.47
#Mann=9,-1,0
  4468.7    0.07       0  4575.8   0.035       0  4599.7    0.07       0
  4969.4    0.05       0  4987.3    0.07       0  5022.8    0.12       0
  5097.9    0.07       0  5235.7   0.035       0  5899.0    0.12       0
Bank Sta=4969.4,4987.3
Exp/Cntr=0.3,0.1

Type RM Length L Ch R = 1,2766,451,451,451
BEGIN DESCRIPTION:
Miller Creek 6.0
END DESCRIPTION:
XS GIS Cut Line= 3
      2165292.68     13861206.06      2166675.00     13860325.00
      2167909.03     13859435.71
#Sta/Elev= 30
  3366.3 1021.15  3381.3 1020.83  3412.7 1018.31  3491.4 1016.83  3571.4 1012.96
  3833.2 1001.37  3977.1  998.51  4036.1  997.59  4096.3  995.26  4215.5  993.28
  4604.3  986.17  4731.3  985.06  4805.6  981.64  4867.6  978.24  4898.0  973.47
  4976.7  971.41  4983.0  969.51  4983.5  969.01  5000.9  969.51  5002.6  971.40
  5012.9  972.73  5019.0  976.27  5051.4  983.22  5078.5  984.79  5628.9  984.03
  5951.6  987.02  6208.9  992.82  6360.3 1000.79  6452.3 1011.51  6526.6 1022.86
#Mann=15,-1,0
  3366.3    0.12       0  3381.3   0.035       0  3571.4    0.07       0
  3833.2   0.035       0  3977.1    0.12       0  4036.1   0.035       0
  4096.3    0.07       0  4215.5   0.035       0  4604.3    0.07       0
  4805.6    0.12       0  4983.0    0.05       0  5000.9    0.12       0
  5051.4    0.07       0  5078.5   0.035       0  6208.9    0.12       0
Bank Sta=4983,5000.9
Exp/Cntr=0.3,0.1

Type RM Length L Ch R = 1,2315,444,444,444
BEGIN DESCRIPTION:
Miller Creek 5.0
END DESCRIPTION:
XS GIS Cut Line= 3
      2165318.11     13861349.17      2166925.00     13860675.00
      2168125.03     13859574.98
#Sta/Elev= 30
  3253.3 1020.05  3453.1 1011.69  3683.4 1001.30  3775.4  999.45  4100.2  994.28
  4208.4  992.56  4698.1  982.74  4751.1  975.26  4780.3  974.17  4822.4  976.59
  4851.6  984.58  4875.4  975.61  4924.4  973.06  4957.5  972.53  5008.1  965.18
  5008.6  964.68  5026.2  965.18  5066.5  971.09  5080.7  979.24  5095.5  981.13
  5127.3  981.89  5272.9  982.52  5289.5  982.63  5739.2  982.51  6101.3  987.49
  6260.0  989.92  6404.6 1001.89  6539.0 1024.84  6581.5 1027.96  6623.8 1028.28
#Mann=15,-1,0
  3253.3   0.035       0  3453.1    0.07       0  3683.4   0.035       0
  3775.4    0.12       0  4100.2    0.07       0  4208.4   0.035       0
  4924.4    0.12       0  5008.1    0.05       0  5026.2    0.12       0
  5095.5    0.07       0  5127.3   0.035       0  5272.9    0.07       0
  5289.5   0.035       0  6101.3    0.07       0  6260.0    0.12       0
Bank Sta=5008.1,5026.2
Exp/Cntr=0.3,0.1

Type RM Length L Ch R = 1,1871,770,770,770
BEGIN DESCRIPTION:
Miller Creek 4.0
END DESCRIPTION:
XS GIS Cut Line= 4
      2165269.77     13861513.65      2167275.00     13860925.00
      2167565.50     13860507.58      2168511.09     13860160.41
#Sta/Elev= 30
  2906.3 1020.93  2933.6 1019.99  3184.1 1008.89  3451.7  999.82  3528.9  998.48
  4046.1  991.07  4339.9  988.16  4586.2  989.98  4756.4  986.67  4940.9  977.81
  4946.1  975.27  4974.2  973.50  4984.5  961.93  4985.0  961.43  5002.6  961.93
  5044.0  963.89  5081.4  963.18  5125.8  977.32  5154.5  979.76  5241.2  980.45
  5653.3  978.79  5726.2  974.45  5842.8  973.93  5958.6  979.74  6081.3  983.30
  6223.1 1006.60  6278.8 1024.70  6420.3 1036.85  6462.9 1045.54  6512.0 1047.90
#Mann=12,-1,0
  2906.3    0.12       0  2933.6   0.035       0  3184.1    0.07       0
  3451.7   0.035       0  3528.9    0.12       0  4046.1    0.07       0
  4339.9   0.035       0  4984.5   0.035       0  5002.6   0.035       0
  5044.0    0.12       0  5241.2   0.035       0  5958.6    0.12       0
Bank Sta=4984.5,5002.6
Exp/Cntr=0.3,0.1

Type RM Length L Ch R = 1,1101,137,137,137
BEGIN DESCRIPTION:
Miller Creek 3.0
END DESCRIPTION:
XS GIS Cut Line= 4
      2165308.48     13861591.81      2167260.34     13861192.55
      2167969.08     13860766.53      2168515.51     13860394.06
#Sta/Elev= 30
  2180.8 1017.63  2368.8 1010.22  2671.3  999.86  2772.5  997.94  3379.8  989.62
  3549.6  989.91  3881.8  995.31  4172.9  986.85  4328.8  988.07  4377.4  982.98
  4414.3  985.58  4604.7  981.20  4837.9  970.08  4902.0  960.74  4916.6  961.67
  4997.2  949.56  4997.7  949.06  5015.5  949.56  5027.3  951.14  5033.4  959.69
  5048.3  965.02  5063.2  963.38  5090.5  968.83  5141.1  974.68  5293.6  979.94
  5344.4  995.09  5416.3 1023.33  5559.9 1033.40  5610.7 1041.64  5661.3 1044.77
#Mann=11,-1,0
  2180.8   0.035       0  2368.8    0.07       0  2671.3   0.035       0
  2772.5    0.12       0  3379.8   0.035       0  3549.6    0.07       0
  3881.8   0.035       0  4916.6    0.07       0  4997.2    0.05       0
  5015.5    0.07       0  5090.5    0.12       0
Bank Sta=4997.2,5015.5
Exp/Cntr=0.3,0.1

Type RM Length L Ch R = 1,964,460,460,460
BEGIN DESCRIPTION:
Miller Creek 2.0
END DESCRIPTION:
XS GIS Cut Line= 4
      2165295.11     13861674.10      2167407.32     13861279.83
      2168089.40     13860823.16      2168589.32     13860504.66
#Sta/Elev= 30
  2031.5 1017.28  2194.8 1010.99  2430.4 1002.89  2531.2 1000.14  2632.1  998.06
  2664.8  997.22  3236.9  990.19  3615.7  993.27  3802.9  993.19  4176.0  979.84
  4401.8  981.25  4444.7  981.08  4860.1  975.93  4968.2  967.18  4994.1  957.88
  5001.0  957.56  5016.3  948.62  5016.8  948.12  5034.6  948.62  5083.1  958.60
  5104.2  966.72  5198.2  980.69  5228.6  992.06  5249.8  991.65  5265.0  998.33
  5286.2 1000.43  5351.5 1022.50  5510.5 1033.76  5562.1 1044.06  5593.8 1045.23
#Mann=14,-1,0
  2031.5   0.035       0  2194.8    0.07       0  2430.4   0.035       0
  2531.2    0.07       0  2632.1   0.035       0  2664.8    0.12       0
  3236.9   0.035       0  3615.7    0.07       0  3802.9   0.035       0
  4401.8    0.07       0  4444.7   0.035       0  4994.1    0.12       0
  5016.3    0.05       0  5034.6    0.12       0
Bank Sta=5016.3,5034.6
Exp/Cntr=0.3,0.1

Type RM Length L Ch R = 1,504,364,364,364
BEGIN DESCRIPTION:
Miller Creek 1.0
END DESCRIPTION:
XS GIS Cut Line= 3
      2165290.31     13861791.09      2168325.00     13861175.00
      2168524.97     13860975.03
#Sta/Elev= 30
  1902.9 1015.98  2019.7 1010.66  2304.5 1002.95  2405.7  999.35  2494.2  997.88
  2661.3  995.26  3113.9  990.56  3605.9  992.75  3695.7  990.79  3814.5  988.50
  3915.8  981.51  4050.5  976.46  4562.5  978.45  4644.9  979.24  4856.6  980.60
  4891.9  978.60  4935.0  975.61  4948.5  971.03  4974.2  952.32  4987.7  946.68
  4988.2  946.18  5006.1  946.68  5013.6  951.80  5041.9  961.61  5056.1  970.14
  5078.3  972.62  5126.8  982.13  5254.1 1039.88  5268.2 1045.52  5282.3 1047.09
#Mann=16,-1,0
  1902.9   0.035       0  2019.7    0.07       0  2304.5   0.035       0
  2405.7    0.12       0  2494.2   0.035       0  2661.3    0.12       0
  3113.9   0.035       0  3605.9    0.07       0  3695.7   0.035       0
  4562.5    0.07       0  4644.9   0.035       0  4891.9    0.12       0
  4935.0    0.12       0  4987.7    0.05       0  5006.1    0.12       0
  5078.3    0.12       0
Bank Sta=4987.7,5006.1
Exp/Cntr=0.3,0.1

Type RM Length L Ch R = 1,140,0,0,0
BEGIN DESCRIPTION:
Miller Creek 0.0
END DESCRIPTION:
XS GIS Cut Line= 3
      2165285.51     13861908.09      2168416.16     13861509.38
      2168660.27     13861094.86
#Sta/Elev= 30
  1850.8 1014.42  1920.9 1009.67  2272.1 1001.26  2381.9  998.42  2746.5  994.03
  2846.3  993.36  2946.0  992.76  3453.1  991.94  3916.8  976.42  4168.9  979.41
  4840.7  976.10  4940.4  966.21  4955.2  963.19  4986.3  947.94  4986.8  947.44
  5004.7  947.94  5010.5  949.27  5016.0  960.98  5031.6  960.88  5037.4  968.61
  5051.8  968.12  5058.9  974.81  5068.7  974.80  5074.5  978.56  5225.9  982.97
  5280.0  984.06  5338.1  984.66  5383.1  986.89  5410.3  994.94  5487.8 1040.03
#Mann=14,-1,0
  1850.8   0.035       0  2272.1    0.12       0  2381.9   0.035       0
  2746.5    0.07       0  2846.3    0.12       0  2946.0   0.035       0
  4840.7    0.12       0  4940.4   0.033       0  4986.3   0.033       0
  5004.7   0.033       0  5051.8    0.12       0  5225.9    0.12       0
  5280.0    0.12       0  5338.1    0.12       0
Bank Sta=4986.3,5004.7
Exp/Cntr=0.3,0.1

Chan Stop Cuts=-1
