--- SWEDE CREEK.prj (project) ---

Proj Title=SWEDE CREEK Base Level Engineering
Current Plan=p01
Default Exp/Contr=0.3,0.1
English Units
Geom File=g01
Flow File=f01
Plan File=p01
Y Axis Title=Elevation
X Axis Title(PF)=Main Channel Distance
X Axis Title(XS)=Station
BEGIN DESCRIPTION:
SWEDE CREEK
END DESCRIPTION:
DSS Export Rating Curves= 0
DSS Export Rating Curve Sorted= 0
DSS Export Volume Flow Curves= 0
DXF OffsetX= 0
DXF OffsetY= 0
DXF ScaleX= 1
DXF ScaleY= 10

--- SWEDE CREEK.p01 (plan) ---

Plan Title=Multiple Run
Short Identifier=Multiple
Geom File=g01
Flow File=f01
Subcritical Flow
K Sum by GR= 0
Std Step Tol= 0.01
Critical Tol= 0.01
Num of Std Step Trials= 20
Max Error Tol= 0.3
Flow Tol Ratio= 0.001
Split Flow NTrial= 30
Split Flow Tol= 0.02
Split Flow Ratio= 0.02
Log Output Level= 0
Friction Slope Method= 1
Unsteady Friction Slope Method= 2
Unsteady Bridges Friction Slope Method= 1
Parabolic Critical Depth
Global Vel Dist=  1 , 1 , 1
Global Log Level= 0
CheckData=True
Encroach Param= -1, 0, 0, 0
BEGIN DESCRIPTION:
Multiple Run
END DESCRIPTION:

--- SWEDE CREEK.f01 (steady flow) ---

Flow Title=Multiple
Program Version=4.10
Number of Profiles= 7
Profile Names=10-year,25-year,50-year,1pct_min,100-year,1pct_plu,500-year
River Rch & RM=SWEDE CREEK,Reach-1         ,21168
    1155    1972    2756    1869    3729    7440    6747
River Rch & RM=SWEDE CREEK,Reach-1         ,18825
    2533    4484    6419    4441    8862   17682   16721
River Rch & RM=SWEDE CREEK,Reach-1         ,12453
    2686    4761    6820    4720    9418   18792   17784
River Rch & RM=SWEDE CREEK,Reach-1         ,9317
    4291    7747   11235    7860   15683   31291   30261
River Rch & RM=SWEDE CREEK,Reach-1         ,1902
    4773    8652   12582    8822   17602   35120   34120
Boundary for River Rch & Prof#=SWEDE CREEK,Reach-1         , 1
Up Type= 0
Dn Type= 3
Dn Slope=0.005
Boundary for River Rch & Prof#=SWEDE CREEK,Reach-1         , 2
Up Type= 0
Dn Type= 3
Dn Slope=0.005
Boundary for River Rch & Prof#=SWEDE CREEK,Reach-1         , 3
Up Type= 0
Dn Type= 3
Dn Slope=0.005
Boundary for River Rch & Prof#=SWEDE CREEK,Reach-1         , 4
Up Type= 0
Dn Type= 3
Dn Slope=0.005
Boundary for River Rch & Prof#=SWEDE CREEK,Reach-1         , 5
Up Type= 0
Dn Type= 3
Dn Slope=0.005
Boundary for River Rch & Prof#=SWEDE CREEK,Reach-1         , 6
Up Type= 0
Dn Type= 3
Dn Slope=0.005
Boundary for River Rch & Prof#=SWEDE CREEK,Reach-1         , 7
Up Type= 0
Dn Type= 3
Dn Slope=0.005
DSS Import GetInterval= 0
DSS Import GetPeak= 0
DSS Import FillOption= 0

--- SWEDE CREEK.g01 (geometry) ---

Geom Title=Existing Conditions

River Reach=SWEDE CREEK,Reach-1
Reach XY= 30
      2101375.00     13852325.00      2101575.46     13852885.19
      2101377.06     13853180.85      2101373.38     13853563.17
      2100775.00     13853825.00      2100766.92     13854428.30
      2100324.41     13855404.95      2100378.08     13855666.70
      2100715.20     13855964.52      2101173.45     13856028.75
      2101421.46     13856276.47      2101273.78     13857514.50
      2100917.12     13858481.16      2100228.54     13859126.47
      2099777.26     13860580.94      2100175.39     13861995.13
      2099724.80     13862705.08      2099988.48     13863238.56
      2100326.55     13863421.25      2101428.34     13863482.99
      2101567.19     13863618.81      2101261.37     13864238.21
      2100804.45     13864444.44      2100426.78     13865018.87
      2100776.47     13865421.45      2101364.39     13865464.94
      2101804.57     13866805.27      2102204.96     13866975.61
      2102523.72     13866828.37      2102675.00     13867175.00

Type RM Length L Ch R = 1,21168,486,486,486
BEGIN DESCRIPTION:
SWEDE CREEK 46.0
END DESCRIPTION:
XS GIS Cut Line= 3
      2100825.03     13852425.00      2101425.00     13852475.00
      2102099.02     13852429.50
#Sta/Elev= 30
  4398.7 1321.58  4438.8 1319.75  4478.9 1315.25  4489.0 1313.34  4519.1 1302.84
  4539.2 1300.48  4576.8 1298.43  4705.2 1296.14  4813.1 1295.92  4955.6 1295.73
  4970.6 1295.25  4988.7 1289.04  4989.0 1288.54  4992.7 1289.04  4998.2 1290.90
  5010.8 1291.42  5050.9 1289.84  5075.4 1292.29  5141.1 1293.90  5161.1 1298.31
  5201.2 1315.93  5238.0 1319.65  5351.5 1324.56  5401.7 1330.00  5431.7 1336.52
  5461.8 1339.83  5518.6 1342.72  5642.2 1346.47  5652.2 1345.82  5676.3 1349.31
#Mann=7,-1,0
  4398.7    0.12       0  4705.2    0.07       0  4813.1    0.12       0
  4955.6    0.07       0  4988.7    0.05       0  4992.7    0.07       0
  5238.0    0.12       0
Bank Sta=4988.7,4992.7
Exp/Cntr=0.3,0.1

Type RM Length L Ch R = 1,20682,473,473,473
BEGIN DESCRIPTION:
SWEDE CREEK 45.0
END DESCRIPTION:
XS GIS Cut Line= 3
      2100975.01     13852475.01      2101575.00     13852875.00
      2102121.71     13852711.24
#Sta/Elev= 30
  4278.5 1298.92  4394.2 1295.06  4503.9 1293.57  4593.2 1293.00  4667.6 1292.19
  4697.6 1293.29  4703.6 1292.42  4775.7 1290.25  4935.0 1286.86  4963.5 1284.80
  4971.0 1285.32  4992.1 1284.26  4996.6 1285.40  5002.2 1285.40  5014.1 1283.51
  5014.4 1283.01  5018.1 1283.51  5030.9 1285.23  5041.3 1290.00  5049.2 1295.26
  5054.4 1295.49  5087.5 1307.58  5093.5 1311.16  5104.0 1313.99  5166.6 1317.52
  5324.8 1320.59  5395.7 1321.62  5406.7 1323.01  5427.6 1322.54  5570.3 1327.97
#Mann=6,-1,0
  4278.5    0.07       0  4503.9    0.12       0  4593.2    0.07       0
  5014.1    0.05       0  5018.1    0.07       0  5324.8    0.12       0
Bank Sta=5014.1,5018.1
Exp/Cntr=0.3,0.1

Type RM Length L Ch R = 1,20209,481,481,481
BEGIN DESCRIPTION:
SWEDE CREEK 44.0
END DESCRIPTION:
XS GIS Cut Line= 3
      2100775.00     13852675.00      2101375.00     13853275.00
      2102015.69     13853453.79
#Sta/Elev= 30
  4151.6 1314.00  4165.7 1312.22  4194.0 1304.08  4236.5 1297.37  4264.7 1295.07
  4377.3 1290.92  4471.4 1288.45  4703.1 1285.20  4731.4 1285.53  4773.9 1284.47
  4802.1 1282.45  4858.7 1281.99  4872.8 1280.90  4957.7 1280.77  4969.8 1278.66
  4970.1 1278.16  4973.8 1278.66  5042.1 1280.65  5090.8 1282.17  5103.9 1281.52
  5169.5 1284.50  5237.8 1285.63  5270.1 1287.27  5301.2 1290.77  5384.3 1294.60
  5503.0 1297.25  5542.4 1299.16  5571.1 1298.91  5642.2 1302.55  5665.3 1304.00
#Mann=7,-1,0
  4151.6    0.07       0  4377.3    0.12       0  4471.4    0.07       0
  4969.8    0.05       0  4973.8    0.07       0  5042.1    0.12       0
  5642.2    0.07       0
Bank Sta=4969.8,4973.8
Exp/Cntr=0.3,0.1

Type RM Length L Ch R = 1,19728,432,432,432
BEGIN DESCRIPTION:
SWEDE CREEK 43.0
END DESCRIPTION:
XS GIS Cut Line= 3
      2100725.02     13853075.03      2101225.00     13853675.00
      2101549.99     13853850.00
#Sta/Elev= 30
  4223.6 1290.42  4273.7 1289.71  4337.5 1287.55  4358.3 1285.67  4372.6 1283.05
  4386.9 1282.28  4500.1 1280.96  4578.3 1280.75  4704.0 1278.17  4728.0 1277.06
  4763.1 1277.86  4777.4 1276.83  4813.6 1277.67  4876.4 1277.65  4919.3 1276.15
  4954.5 1274.71  4960.3 1271.97  4960.5 1271.47  4964.3 1271.97  4968.8 1274.63
  4983.1 1275.28  4990.9 1274.07  5007.4 1274.43  5018.4 1280.21  5027.3 1282.27
  5040.3 1282.76  5056.5 1285.53  5094.6 1288.71  5220.4 1291.50  5373.7 1295.99
#Mann=6,-1,0
  4223.6    0.07       0  4500.1    0.12       0  4704.0   0.035       0
  4813.6    0.12       0  4960.3    0.05       0  4964.3    0.12       0
Bank Sta=4960.3,4964.3
Exp/Cntr=0.3,0.1

Type RM Length L Ch R = 1,19296,471,471,471
BEGIN DESCRIPTION:
SWEDE CREEK 42.0
END DESCRIPTION:
XS GIS Cut Line= 3
      2100725.01     13853175.04      2100825.00     13853775.00
      2101144.17     13853915.60
#Sta/Elev= 30
  4392.2 1288.05  4412.4 1287.00  4442.8 1282.50  4493.5 1279.79  4520.4 1279.41
  4668.4 1278.29  4716.6 1276.97  4724.2 1275.76  4729.2 1276.39  4747.0 1274.96
  4770.0 1274.86  4790.3 1273.97  4899.1 1273.00  4929.5 1271.20  4959.9 1271.38
  4970.6 1270.63  4978.2 1268.46  4978.4 1267.96  4982.2 1268.46  4997.9 1271.14
  5022.3 1272.44  5111.7 1272.65  5131.5 1274.03  5160.3 1277.53  5183.6 1278.97
  5206.9 1278.60  5219.0 1279.89  5229.9 1279.07  5264.5 1279.87  5349.2 1283.32
#Mann=8,-1,0
  4392.2    0.07       0  4520.4    0.12       0  4770.0    0.07       0
  4790.3   0.035       0  4970.6    0.07       0  4978.2    0.05       0
  4982.2    0.07       0  5111.7    0.12       0
Bank Sta=4978.2,4982.2
Exp/Cntr=0.3,0.1

Type RM Length L Ch R = 1,18825,460,460,460
BEGIN DESCRIPTION:
SWEDE CREEK 41.0
END DESCRIPTION:
XS GIS Cut Line= 3
      2099975.02     13854175.00      2100775.00     13854225.00
      2101175.04     13854024.98
#Sta/Elev= 30
  4202.9 1284.43  4221.3 1283.79  4253.0 1282.20  4263.0 1282.71  4280.5 1280.24
  4319.9 1277.20  4533.5 1271.41  4713.9 1268.85  4854.1 1269.28  4884.2 1268.03
  4914.3 1268.44  4944.3 1267.35  4954.3 1268.49  4984.4 1268.10  5007.2 1269.34
  5018.4 1268.15  5024.0 1266.24  5024.5 1265.74  5029.2 1265.74  5029.6 1266.24
  5035.2 1266.98  5040.8 1266.79  5049.2 1269.52  5093.9 1268.68  5138.6 1270.22
  5242.0 1272.30  5264.4 1273.63  5309.1 1278.91  5420.9 1281.70  5451.7 1283.31
#Mann=5,-1,0
  4202.9    0.12       0  4221.3   0.035       0  4319.9    0.12       0
  5024.0    0.05       0  5029.6    0.12       0
Bank Sta=5024,5029.6
Exp/Cntr=0.3,0.1

Type RM Length L Ch R = 1,18365,466,466,466
BEGIN DESCRIPTION:
SWEDE CREEK 40.0
END DESCRIPTION:
XS GIS Cut Line= 3
      2100213.65     13854492.00      2100675.00     13854625.00
      2101099.08     13854693.39
#Sta/Elev= 30
  4515.5 1270.63  4636.4 1267.72  4673.0 1266.99  4704.2 1265.13  4722.4 1265.74
  4735.5 1264.39  4777.1 1262.86  4797.1 1260.20  4828.6 1257.49  4846.9 1257.34
  4867.4 1257.52  4872.6 1256.64  4881.2 1257.21  4905.4 1255.20  4922.8 1258.74
  4945.1 1259.16  4964.4 1258.23  4973.6 1257.45  4993.0 1252.97  4998.2 1252.97
  5013.1 1249.17  5013.5 1248.67  5018.7 1249.17  5036.2 1254.07  5046.3 1261.05
  5056.4 1265.11  5066.5 1265.98  5157.7 1269.65  5319.8 1273.14  5425.2 1274.26
#Mann=6,-1,0
  4515.5    0.07       0  4636.4    0.12       0  4797.1    0.07       0
  4846.9    0.12       0  5013.1    0.05       0  5018.7    0.12       0
Bank Sta=5013.1,5018.7
Exp/Cntr=0.3,0.1

Type RM Length L Ch R = 1,17899,295,295,295
BEGIN DESCRIPTION:
SWEDE CREEK 39.0
END DESCRIPTION:
XS GIS Cut Line= 3
      2100075.00     13854825.00      2100425.00     13854975.00
      2100875.03     13854874.99
#Sta/Elev= 30
  4613.8 1273.77  4646.4 1273.49  4675.5 1268.38  4690.0 1268.31  4699.0 1265.31
  4704.5 1266.49  4722.6 1264.02  4798.8 1259.84  4827.8 1256.93  4927.5 1254.02
  4985.5 1251.16  5016.0 1251.00  5016.5 1250.50  5021.8 1251.00  5056.1 1251.54
  5067.6 1253.27  5086.8 1252.15  5106.0 1252.42  5117.5 1251.06  5127.8 1252.94
  5139.1 1253.51  5148.3 1254.47  5154.7 1257.12  5159.8 1256.18  5168.7 1258.29
  5209.7 1261.50  5281.4 1264.03  5363.4 1264.53  5436.4 1267.29  5455.6 1267.31
#Mann=4,-1,0
  4613.8    0.07       0  5016.0    0.05       0  5021.8    0.07       0
  5139.1    0.12       0
Bank Sta=5016,5021.8
Exp/Cntr=0.3,0.1

Type RM Length L Ch R = 1,17604,565,565,565
BEGIN DESCRIPTION:
SWEDE CREEK 38.0
END DESCRIPTION:
XS GIS Cut Line= 2
      2099863.16     13855320.58      2100758.15     13855199.86
#Sta/Elev= 30
  4483.3 1279.21  4561.6 1276.75  4616.3 1275.83  4707.1 1271.83  4712.1 1271.45
  4717.2 1269.47  4737.4 1259.43  4747.5 1256.41  4757.6 1254.65  4767.7 1253.65
  4818.1 1252.06  4862.7 1251.76  4949.3 1250.12  4969.5 1247.48  4979.6 1247.51
  4996.8 1245.99  4997.3 1245.49  5002.2 1245.49  5002.7 1245.99  5008.1 1247.54
  5020.0 1247.79  5030.0 1247.08  5085.8 1250.34  5110.8 1250.43  5191.5 1252.94
  5252.0 1256.50  5272.2 1256.21  5322.7 1258.28  5373.1 1258.67  5386.4 1258.21
#Mann=4,-1,0
  4483.3   0.035       0  4862.7    0.07       0  4996.8    0.05       0
  5002.7    0.07       0
Bank Sta=4996.8,5002.7
Exp/Cntr=0.3,0.1

Type RM Length L Ch R = 1,17039,426,426,426
BEGIN DESCRIPTION:
SWEDE CREEK 37.0
END DESCRIPTION:
XS GIS Cut Line= 3
      2099949.75     13855884.35      2100475.00     13855725.00
      2100675.00     13855325.00
#Sta/Elev= 30
  4450.9 1278.16  4517.6 1276.84  4605.8 1275.02  4671.6 1271.69  4694.1 1271.64
  4749.0 1270.16  4790.8 1267.70  4808.4 1264.98  4846.5 1261.74  4863.9 1258.41
  4912.3 1255.33  4917.5 1255.73  4945.2 1249.80  4958.0 1243.52  4967.5 1240.55
  4980.3 1238.03  4980.8 1237.53  4986.3 1238.03  4989.3 1238.06  4997.2 1240.60
  5052.9 1244.74  5097.6 1243.57  5120.0 1244.11  5178.7 1247.91  5187.1 1247.29
  5237.4 1248.33  5259.7 1249.98  5321.2 1249.16  5409.7 1252.72  5447.0 1254.03
#Mann=7,-1,0
  4450.9    0.07       0  4517.6   0.035       0  4694.1    0.07       0
  4967.5    0.12       0  4980.3    0.05       0  4986.3    0.12       0
  5409.7    0.07       0
Bank Sta=4980.3,4986.3
Exp/Cntr=0.3,0.1

Type RM Length L Ch R = 1,16613,441,441,441
BEGIN DESCRIPTION:
SWEDE CREEK 36.0
END DESCRIPTION:
XS GIS Cut Line= 2
      2100688.28     13856212.40      2101133.64     13855259.65
#Sta/Elev= 30
  4738.2 1245.39  4880.6 1244.33  4923.0 1243.26  4975.5 1236.13  4981.1 1236.16
  4989.2 1238.02  5021.2 1237.35  5030.4 1236.05  5030.9 1235.55  5036.4 1236.05
  5049.6 1237.76  5078.0 1238.48  5095.3 1240.25  5132.7 1240.85  5141.0 1241.79
  5232.1 1242.45  5260.7 1243.89  5357.6 1245.78  5441.8 1248.50  5449.0 1248.13
  5454.5 1249.07  5471.9 1249.81  5540.4 1251.37  5683.0 1257.61  5711.4 1259.95
  5717.8 1261.25  5734.2 1261.41  5739.8 1262.62  5750.9 1263.38  5789.9 1264.72
#Mann=4,-1,0
  4738.2    0.07       0  4880.6    0.12       0  5030.4    0.05       0
  5036.4    0.12       0
Bank Sta=5030.4,5036.4
Exp/Cntr=0.3,0.1

Type RM Length L Ch R = 1,16172,535,535,535
BEGIN DESCRIPTION:
SWEDE CREEK 35.0
END DESCRIPTION:
XS GIS Cut Line= 3
      2100821.23     13856245.49      2101199.75     13856064.91
      2102060.44     13855780.33
#Sta/Elev= 30
  4567.8 1243.66  4871.1 1239.64  4975.9 1232.43  4981.8 1230.22  4992.7 1230.40
  5029.1 1225.18  5029.6 1224.68  5035.2 1225.18  5063.9 1229.62  5069.1 1232.49
  5095.6 1227.09  5100.8 1232.73  5108.9 1229.70  5119.1 1230.85  5127.3 1235.66
  5132.6 1234.55  5159.0 1238.77  5317.7 1255.32  5418.1 1259.51  5456.1 1265.96
  5513.3 1268.31  5561.5 1274.06  5719.5 1277.63  5751.1 1280.23  5767.1 1284.66
  5772.4 1283.13  5782.6 1285.71  5798.8 1286.88  5867.5 1287.63  5893.7 1290.81
#Mann=4,-1,0
  4567.8    0.07       0  5029.1    0.05       0  5035.2    0.07       0
  5108.9    0.12       0
Bank Sta=5029.1,5035.2
Exp/Cntr=0.3,0.1

Type RM Length L Ch R = 1,15637,438,438,438
BEGIN DESCRIPTION:
SWEDE CREEK 34.0
END DESCRIPTION:
XS GIS Cut Line= 3
      2101029.63     13856419.08      2101375.00     13856475.00
      2101668.52     13856478.11
#Sta/Elev= 30
  4645.5 1239.47  4723.3 1237.72  4752.2 1236.88  4771.9 1237.00  4777.0 1236.25
  4833.3 1234.87  4843.7 1234.15  4883.9 1229.94  4894.1 1228.31  4900.3 1225.89
  4914.3 1223.89  4934.6 1223.15  4962.0 1220.75  4967.1 1220.90  4975.1 1219.60
  4985.2 1216.74  4989.5 1213.85  4990.0 1213.35  4995.6 1213.35  4996.1 1213.85
  5005.4 1214.25  5015.4 1229.94  5025.4 1235.47  5055.4 1240.27  5115.4 1251.62
  5145.4 1256.14  5215.4 1259.51  5225.4 1260.28  5245.4 1263.09  5288.9 1264.80
#Mann=4,-1,0
  4645.5    0.07       0  4723.3    0.12       0  4989.5    0.05       0
  4996.1    0.12       0
Bank Sta=4989.5,4996.1
Exp/Cntr=0.3,0.1

Type RM Length L Ch R = 1,15199,481,481,481
BEGIN DESCRIPTION:
SWEDE CREEK 33.0
END DESCRIPTION:
XS GIS Cut Line= 3
      2101175.02     13856875.00      2101275.00     13856875.00
      2101567.80     13856811.44
#Sta/Elev= 30
  4900.0 1231.95  4930.0 1228.11  4950.0 1223.59  4970.0 1215.85  4980.0 1209.97
  4986.6 1207.58  4987.1 1207.08  4992.8 1207.08  4993.3 1207.58  4997.5 1209.46
  5002.5 1209.46  5010.2 1212.47  5019.4 1212.35  5030.7 1213.17  5051.1 1216.10
  5061.4 1218.67  5068.6 1221.15  5073.7 1220.83  5081.8 1224.58  5117.7 1234.01
  5122.9 1233.67  5133.0 1235.50  5173.9 1239.16  5194.4 1239.65  5210.9 1240.85
  5255.0 1242.68  5266.0 1244.17  5276.3 1244.65  5286.5 1245.91  5299.6 1245.73
#Mann=3,-1,0
  4900.0    0.12       0  4986.6    0.05       0  4993.3    0.12       0
Bank Sta=4986.6,4993.3
Exp/Cntr=0.3,0.1

Type RM Length L Ch R = 1,14718,484,484,484
BEGIN DESCRIPTION:
SWEDE CREEK 32.0
END DESCRIPTION:
XS GIS Cut Line= 3
      2100866.38     13857280.19      2101275.00     13857325.00
      2101658.11     13857328.80
#Sta/Elev= 30
  4593.8 1234.04  4680.9 1234.00  4685.9 1233.13  4693.0 1233.58  4785.5 1232.30
  4803.7 1232.02  4868.2 1229.00  4874.1 1227.65  4894.2 1225.59  4924.4 1219.51
  4944.5 1208.68  4954.3 1205.65  4964.6 1206.71  4974.7 1206.78  4981.3 1205.45
  4981.8 1204.95  4987.6 1204.95  4988.1 1205.45  5007.4 1205.78  5024.9 1207.70
  5034.9 1212.11  5044.9 1217.84  5054.9 1220.46  5094.9 1228.28  5114.9 1231.03
  5174.9 1234.47  5194.9 1236.28  5244.9 1238.35  5264.9 1240.69  5388.0 1243.43
#Mann=4,-1,0
  4593.8    0.07       0  4785.5    0.12       0  4981.3    0.05       0
  4988.1    0.12       0
Bank Sta=4981.3,4988.1
Exp/Cntr=0.3,0.1

Type RM Length L Ch R = 1,14234,466,466,466
BEGIN DESCRIPTION:
SWEDE CREEK 31.0
END DESCRIPTION:
XS GIS Cut Line= 3
      2100800.43     13857637.82      2101175.00     13857775.00
      2101660.75     13857787.11
#Sta/Elev= 30
  4601.1 1229.83  4680.5 1229.13  4701.8 1227.86  4720.8 1227.80  4756.6 1225.26
  4781.8 1226.37  4850.9 1225.20  4868.0 1223.70  4898.5 1219.12  4904.2 1215.94
  4923.7 1210.38  4936.1 1205.91  4954.2 1202.58  4984.7 1200.28  4990.1 1199.45
  4993.9 1197.59  4994.4 1197.09  5000.8 1197.59  5010.0 1200.38  5020.0 1201.09
  5030.0 1205.21  5040.0 1212.38  5050.0 1217.79  5060.0 1220.83  5100.0 1227.82
  5150.0 1231.18  5290.1 1235.39  5310.1 1234.91  5410.1 1236.65  5485.9 1236.65
#Mann=3,-1,0
  4601.1    0.12       0  4993.9    0.05       0  5000.8    0.12       0
Bank Sta=4993.9,5000.8
Exp/Cntr=0.3,0.1

Type RM Length L Ch R = 1,13768,456,456,456
BEGIN DESCRIPTION:
SWEDE CREEK 30.0
END DESCRIPTION:
XS GIS Cut Line= 3
      2100658.13     13858051.04      2100975.00     13858175.00
      2101890.34     13857992.07
#Sta/Elev= 30
  4654.6 1226.31  4841.5 1224.42  4955.5 1220.56  4985.3 1205.48  4992.2 1199.23
  4997.4 1199.23  5011.8 1192.67  5012.3 1192.17  5018.7 1192.67  5020.4 1194.42
  5035.6 1194.27  5076.5 1198.10  5096.8 1205.01  5122.4 1211.29  5127.5 1211.05
  5173.4 1220.59  5219.2 1223.01  5239.6 1225.74  5331.5 1228.18  5479.4 1226.84
  5606.7 1231.32  5688.6 1232.04  5729.1 1230.22  5739.6 1231.93  5785.5 1230.46
  5800.5 1232.60  5841.6 1233.08  5861.7 1230.39  5892.6 1234.40  5928.3 1235.78
#Mann=3,-1,0
  4654.6    0.12       0  5011.8    0.05       0  5018.7    0.12       0
Bank Sta=5011.8,5018.7
Exp/Cntr=0.3,0.1

Type RM Length L Ch R = 1,13312,413,413,413
BEGIN DESCRIPTION:
SWEDE CREEK 29.0
END DESCRIPTION:
XS GIS Cut Line= 3
      2100439.35     13857891.33      2100825.00     13858575.00
      2101900.59     13858898.08
#Sta/Elev= 30
  4210.7 1223.62  4226.4 1221.93  4269.8 1221.50  4329.1 1223.22  4334.8 1224.45
  4415.7 1225.18  4534.2 1223.46  4570.8 1224.48  4641.1 1222.42  4647.8 1222.23
  4717.6 1220.58  4834.9 1213.30  4885.1 1204.98  4981.9 1196.00  4992.8 1192.47
  5012.2 1190.26  5013.5 1188.72  5014.0 1188.22  5021.2 1188.72  5050.4 1190.03
  5068.7 1193.04  5078.2 1196.57  5089.6 1203.79  5121.7 1214.42  5182.6 1219.74
  5350.6 1226.27  5475.9 1229.04  5590.8 1230.22  5600.0 1229.23  6118.7 1242.89
#Mann=5,-1,0
  4210.7    0.12       0  4641.1    0.07       0  4647.8    0.12       0
  5013.5    0.05       0  5021.2    0.12       0
Bank Sta=5013.5,5021.2
Exp/Cntr=0.3,0.1

Type RM Length L Ch R = 1,12899,446,446,446
BEGIN DESCRIPTION:
SWEDE CREEK 28.0
END DESCRIPTION:
XS GIS Cut Line= 3
      2100424.99     13858724.99      2100575.00     13858875.00
      2101011.15     13858984.77
#Sta/Elev= 30
  4795.8 1209.13  4824.1 1206.78  4852.4 1202.64  4880.7 1195.67  4909.0 1190.68
  4937.2 1188.04  4951.4 1187.52  4965.5 1185.83  4975.8 1180.39  4976.3 1179.89
  4983.0 1179.89  4983.5 1180.39  4993.8 1185.31  5001.7 1190.32  5004.4 1192.03
  5010.5 1192.03  5025.9 1197.41  5043.4 1199.67  5067.0 1201.88  5100.8 1203.92
  5121.4 1203.78  5131.7 1205.13  5162.6 1210.96  5190.4 1213.61  5265.7 1215.87
  5313.7 1218.73  5368.9 1220.10  5395.9 1221.90  5443.0 1223.01  5457.7 1224.33
#Mann=6,-1,0
  4795.8    0.07       0  4975.8    0.05       0  4983.5    0.07       0
  5001.7   0.035       0  5043.4    0.07       0  5443.0    0.12       0
Bank Sta=4975.8,4983.5
Exp/Cntr=0.3,0.1

Type RM Length L Ch R = 1,12453,463,463,463
BEGIN DESCRIPTION:
SWEDE CREEK 27.0
END DESCRIPTION:
XS GIS Cut Line= 3
      2099956.66     13858988.51      2100225.00     13859125.00
      2100876.83     13859373.94
#Sta/Elev= 30
  4695.1 1227.20  4720.9 1225.51  4749.3 1221.46  4848.7 1216.52  4876.6 1213.41
  4893.2 1209.38  4965.6 1203.85  4982.2 1188.94  4987.8 1187.72  4993.4 1181.43
  4998.8 1181.43  5001.7 1178.01  5002.2 1177.51  5009.9 1178.01  5017.6 1181.12
  5035.9 1183.79  5071.3 1184.84  5111.1 1189.11  5120.8 1190.02  5167.4 1190.04
  5175.6 1191.07  5215.4 1192.22  5253.1 1195.12  5295.9 1201.67  5338.7 1203.90
  5400.1 1211.38  5442.5 1214.07  5576.8 1218.16  5617.0 1219.93  5693.9 1221.56
#Mann=7,-1,0
  4695.1    0.12       0  5001.7    0.05       0  5009.9    0.12       0
  5111.1   0.035       0  5215.4    0.07       0  5442.5    0.12       0
  5576.8    0.07       0
Bank Sta=5001.7,5009.9
Exp/Cntr=0.3,0.1

Type RM Length L Ch R = 1,11990,450,450,450
BEGIN DESCRIPTION:
SWEDE CREEK 26.0
END DESCRIPTION:
XS GIS Cut Line= 3
      2099790.03     13859360.05      2100175.00     13859575.00
      2100585.19     13859769.78
#Sta/Elev= 30
  4563.2 1219.68  4600.8 1219.11  4637.6 1217.11  4725.4 1207.87  4752.8 1206.25
  4763.0 1206.69  4784.8 1204.68  4843.8 1195.25  4865.9 1189.92  4907.7 1186.78
  4923.9 1185.84  4936.7 1183.55  4946.8 1178.70  4952.7 1177.43  4970.3 1177.42
  4970.8 1176.92  4978.6 1177.42  4996.1 1177.98  5012.7 1180.14  5048.4 1180.26
  5080.9 1183.62  5086.4 1183.37  5109.2 1187.64  5114.8 1190.44  5137.4 1196.54
  5160.1 1200.07  5214.4 1204.85  5258.7 1206.24  5322.2 1211.69  5458.2 1216.15
#Mann=5,-1,0
  4563.2    0.12       0  4907.7    0.07       0  4970.3    0.05       0
  4978.6    0.07       0  5322.2    0.12       0
Bank Sta=4970.3,4978.6
Exp/Cntr=0.3,0.1

Type RM Length L Ch R = 1,11540,447,447,447
BEGIN DESCRIPTION:
SWEDE CREEK 25.0
END DESCRIPTION:
XS GIS Cut Line= 3
      2099553.90     13859741.99      2100025.00     13859975.00
      2100505.34     13860026.72
#Sta/Elev= 30
  4469.6 1218.78  4538.1 1216.02  4577.4 1213.01  4582.9 1213.25  4605.4 1210.44
  4622.2 1206.26  4727.4 1201.14  4756.8 1196.89  4762.4 1196.91  4779.3 1191.45
  4824.1 1184.06  4913.9 1179.68  4958.7 1174.46  4997.7 1173.40  5010.6 1172.21
  5011.1 1172.20  5011.6 1171.70  5019.5 1172.20  5035.4 1173.90  5046.2 1182.45
  5065.6 1193.55  5085.7 1197.16  5133.1 1201.59  5236.6 1204.22  5246.6 1205.95
  5286.9 1209.72  5317.0 1210.37  5414.0 1214.88  5419.1 1214.34  5478.3 1215.64
#Mann=4,-1,0
  4469.6    0.12       0  5010.6    0.07       0  5011.1    0.05       0
  5019.5    0.07       0
Bank Sta=5011.1,5019.5
Exp/Cntr=0.3,0.1

Type RM Length L Ch R = 1,11093,481,481,481
BEGIN DESCRIPTION:
SWEDE CREEK 24.0
END DESCRIPTION:
XS GIS Cut Line= 3
      2099625.05     13860375.00      2099875.00     13860375.00
      2100460.07     13860273.26
#Sta/Elev= 30
  4754.7 1212.68  4774.7 1208.91  4804.7 1201.29  4834.7 1198.35  4844.7 1196.25
  4854.7 1192.87  4874.7 1182.51  4894.7 1174.96  4904.7 1172.17  4932.1 1172.02
  4944.7 1171.06  4964.7 1171.32  4994.7 1170.29  4998.0 1169.56  4998.5 1169.06
  5006.4 1169.56  5025.0 1172.33  5031.9 1174.37  5037.0 1174.05  5045.3 1176.27
  5055.4 1177.38  5105.3 1180.26  5116.3 1180.92  5146.1 1186.10  5177.2 1188.98
  5327.6 1197.18  5379.6 1197.59  5431.0 1200.79  5552.8 1204.59  5598.5 1208.33
#Mann=6,-1,0
  4754.7    0.12       0  4932.1    0.07       0  4998.0    0.05       0
  5006.4    0.07       0  5105.3   0.035       0  5327.6    0.07       0
Bank Sta=4998,5006.4
Exp/Cntr=0.3,0.1

Type RM Length L Ch R = 1,10612,482,482,482
BEGIN DESCRIPTION:
SWEDE CREEK 23.0
END DESCRIPTION:
XS GIS Cut Line= 3
      2099512.25     13860783.66      2099775.00     13860825.00
      2100660.77     13860634.52
#Sta/Elev= 30
  4729.8 1207.55  4769.3 1202.35  4864.2 1198.78  4904.7 1196.12  4924.9 1196.23
  4945.2 1194.52  4955.3 1191.84  4962.0 1187.16  4967.0 1187.29  4985.7 1176.17
  4993.3 1168.64  4998.3 1168.64  5009.8 1164.39  5011.1 1163.94  5011.6 1163.44
  5019.5 1163.94  5114.1 1170.94  5179.9 1173.74  5262.1 1174.71  5415.2 1184.01
  5449.3 1186.94  5476.5 1193.22  5493.5 1195.52  5592.3 1199.19  5630.0 1202.55
  5701.6 1204.65  5735.2 1206.36  5748.8 1208.31  5803.8 1212.46  5901.8 1215.03
#Mann=5,-1,0
  4729.8    0.12       0  5009.8    0.07       0  5011.1    0.05       0
  5019.5    0.07       0  5748.8    0.12       0
Bank Sta=5011.1,5019.5
Exp/Cntr=0.3,0.1

Type RM Length L Ch R = 1,10130,385,385,385
BEGIN DESCRIPTION:
SWEDE CREEK 22.0
END DESCRIPTION:
XS GIS Cut Line= 3
      2099575.02     13861125.01      2099875.00     13861275.00
      2100691.38     13860978.62
#Sta/Elev= 30
  4660.5 1193.21  4696.8 1190.32  4727.6 1184.25  4805.2 1179.36  4965.1 1170.42
  4981.9 1166.22  4987.5 1166.55  4993.1 1163.46  4998.5 1163.46  5001.6 1161.57
  5002.1 1161.07  5010.1 1161.57  5041.8 1163.92  5091.6 1164.58  5103.0 1167.38
  5123.0 1168.50  5272.8 1170.68  5347.0 1179.73  5474.4 1185.58  5479.7 1187.44
  5505.0 1186.14  5510.3 1188.18  5535.6 1187.56  5591.5 1191.25  5596.8 1193.95
  5627.4 1196.16  5771.8 1203.13  5806.6 1204.55  5831.0 1207.94  5864.4 1209.35
#Mann=7,-1,0
  4660.5    0.12       0  4805.2   0.035       0  5001.6   0.035       0
  5010.1   0.035       0  5272.8    0.07       0  5771.8    0.12       0
  5806.6    0.07       0
Bank Sta=5001.6,5010.1
Exp/Cntr=0.3,0.1

Type RM Length L Ch R = 1,9745,428,428,428
BEGIN DESCRIPTION:
SWEDE CREEK 21.0
END DESCRIPTION:
XS GIS Cut Line= 3
      2099574.58     13861196.29      2099933.96     13861613.41
      2100500.33     13861567.60
#Sta/Elev= 30
  4357.7 1191.36  4378.6 1189.26  4399.4 1184.16  4413.7 1182.62  4477.3 1178.77
  4534.4 1177.38  4548.6 1175.89  4633.2 1172.21  4810.8 1169.81  4875.6 1167.36
  4935.9 1166.52  4959.5 1166.06  4969.5 1163.79  4975.3 1159.80  4975.8 1159.30
  4983.9 1159.80  5009.7 1161.71  5029.7 1161.11  5120.0 1165.00  5210.3 1167.12
  5230.4 1171.16  5260.5 1182.01  5290.6 1187.36  5310.6 1192.31  5319.2 1195.47
  5324.2 1193.98  5330.7 1196.73  5340.7 1198.51  5431.4 1201.54  5476.5 1203.01
#Mann=6,-1,0
  4357.7    0.12       0  4875.6    0.07       0  4935.9    0.12       0
  4975.3    0.05       0  4983.9    0.12       0  5431.4   0.035       0
Bank Sta=4975.3,4983.9
Exp/Cntr=0.3,0.1

Type RM Length L Ch R = 1,9317,538,538,538
BEGIN DESCRIPTION:
SWEDE CREEK 20.0
END DESCRIPTION:
XS GIS Cut Line= 3
      2098818.33     13862233.10      2100067.32     13861980.15
      2100679.96     13861955.14
#Sta/Elev= 30
  3617.4 1209.41  3670.3 1206.27  3960.1 1199.92  4001.4 1199.14  4063.2 1197.35
  4114.0 1192.90  4144.6 1186.92  4226.2 1179.65  4256.8 1169.93  4297.6 1161.34
  4438.0 1157.71  4438.5 1157.21  4446.6 1157.71  4493.0 1160.16  4538.6 1158.35
  4543.7 1160.67  4552.7 1161.27  4675.1 1158.99  4858.8 1164.27  4894.9 1161.29
  4949.5 1161.43  4959.5 1159.80  5009.5 1158.50  5029.3 1160.14  5049.6 1166.86
  5079.6 1185.10  5109.6 1199.66  5169.3 1202.40  5212.4 1203.22  5504.9 1204.91
#Mann=10,-1,0
  3617.4    0.07       0  3670.3   0.035       0  3960.1    0.07       0
  4001.4    0.12       0  4063.2    0.07       0  4438.0    0.05       0
  4446.6    0.07       0  5029.3    0.12       0  5169.3   0.035       0
  5212.4    0.07       0
Bank Sta=4438,4446.6
Exp/Cntr=0.3,0.1

Type RM Length L Ch R = 1,8779,477,477,477
BEGIN DESCRIPTION:
SWEDE CREEK 19.0
END DESCRIPTION:
XS GIS Cut Line= 3
      2099046.79     13862334.63      2099925.00     13862425.00
      2100137.26     13862443.38
#Sta/Elev= 30
  4112.3 1205.21  4172.0 1203.57  4251.2 1199.37  4301.5 1189.21  4355.8 1183.87
  4392.0 1173.23  4462.6 1164.09  4495.6 1163.13  4623.2 1161.37  4693.6 1153.00
  4733.8 1152.23  4743.8 1150.29  4754.9 1143.20  4763.9 1142.79  4794.1 1150.97
  4833.8 1152.40  4884.6 1149.54  4924.8 1154.36  4948.1 1150.53  4975.0 1150.72
  4985.1 1148.67  4988.2 1131.12  4988.7 1130.62  4997.0 1131.12  5025.3 1148.59
  5056.7 1156.25  5145.7 1161.60  5175.8 1166.05  5203.9 1163.92  5208.2 1163.96
#Mann=8,-1,0
  4112.3   0.035       0  4172.0    0.07       0  4355.8    0.12       0
  4495.6    0.07       0  4833.8    0.12       0  4988.2    0.05       0
  4997.0    0.12       0  5203.9    0.07       0
Bank Sta=4988.2,4997
Exp/Cntr=0.3,0.1

Type RM Length L Ch R = 1,8302,426,426,426
BEGIN DESCRIPTION:
SWEDE CREEK 18.0
END DESCRIPTION:
XS GIS Cut Line= 3
      2099575.02     13862924.98      2099775.00     13862775.00
      2100091.10     13862787.09
#Sta/Elev= 30
  4754.8 1190.88  4768.3 1190.50  4782.9 1188.38  4791.2 1184.77  4797.5 1183.41
  4812.1 1174.25  4818.3 1173.23  4841.2 1165.92  4862.1 1161.94  4897.5 1159.61
  4911.0 1156.47  4932.9 1144.40  4941.2 1138.12  4947.5 1126.96  4954.8 1125.80
  4968.3 1126.68  4990.1 1125.70  4990.6 1125.20  5004.9 1125.70  5024.8 1125.86
  5044.8 1128.75  5094.8 1132.78  5104.8 1141.52  5124.9 1145.84  5132.7 1150.26
  5137.7 1148.93  5144.9 1152.03  5214.9 1156.77  5259.9 1157.55  5321.1 1157.89
#Mann=4,-1,0
  4754.8   0.035       0  4990.1    0.05       0  5004.9   0.035       0
  5259.9    0.07       0
Bank Sta=4990.1,5004.9
Exp/Cntr=0.3,0.1

Type RM Length L Ch R = 1,7876,463,463,463
BEGIN DESCRIPTION:
SWEDE CREEK 17.0
END DESCRIPTION:
XS GIS Cut Line= 3
      2099775.01     13863274.99      2099925.00     13863125.00
      2100189.36     13862926.00
#Sta/Elev= 30
  4788.0 1190.14  4791.5 1190.14  4816.3 1185.99  4844.6 1172.74  4872.8 1163.42
  4887.0 1160.72  4915.3 1158.42  4929.4 1155.45  4957.7 1133.11  4971.8 1125.92
  4986.0 1123.63  5000.0 1122.82  5000.5 1122.32  5014.9 1122.82  5028.2 1126.09
  5036.5 1126.19  5042.8 1125.31  5086.5 1125.04  5092.8 1125.40  5102.9 1128.11
  5107.4 1129.00  5128.2 1136.44  5157.3 1149.92  5163.6 1151.16  5171.9 1151.85
  5178.2 1153.27  5186.5 1153.16  5192.7 1154.07  5278.4 1156.01  5331.0 1156.31
#Mann=5,-1,0
  4788.0   0.035       0  5000.0   0.035       0  5014.9   0.035       0
  5102.9    0.12       0  5278.4    0.07       0
Bank Sta=5000,5014.9
Exp/Cntr=0.3,0.1

Type RM Length L Ch R = 1,7413,469,469,469
BEGIN DESCRIPTION:
SWEDE CREEK 16.0
END DESCRIPTION:
XS GIS Cut Line= 3
      2100125.02     13863574.97      2100275.00     13863375.00
      2100325.00     13863175.02
#Sta/Elev= 30
  4754.8 1188.34  4769.6 1187.33  4782.9 1186.26  4804.8 1180.75  4832.9 1169.31
  4847.5 1164.94  4862.1 1161.75  4882.9 1159.97  4891.2 1157.10  4897.5 1151.04
  4904.8 1142.16  4912.1 1130.70  4926.6 1124.56  4954.6 1119.63  4955.1 1119.13
  4969.5 1119.63  4991.2 1120.28  4997.5 1121.83  5001.6 1124.48  5015.1 1126.26
  5035.7 1128.00  5064.0 1128.43  5069.2 1130.98  5087.2 1134.43  5097.5 1137.94
  5118.1 1153.76  5159.4 1154.94  5180.0 1151.10  5185.9 1151.27  5210.9 1151.97
#Mann=5,-1,0
  4754.8   0.035       0  4769.6    0.12       0  4954.6    0.05       0
  4969.5    0.12       0  5185.9   0.035       0
Bank Sta=4954.6,4969.5
Exp/Cntr=0.3,0.1

Type RM Length L Ch R = 1,6944,453,453,453
BEGIN DESCRIPTION:
SWEDE CREEK 15.0
END DESCRIPTION:
XS GIS Cut Line= 3
      2100460.19     13863787.10      2100725.00     13863425.00
      2100725.00     13863225.00
#Sta/Elev= 30
  4551.0 1169.36  4571.9 1168.84  4578.4 1169.51  4584.6 1167.76  4599.2 1170.35
  4620.1 1164.53  4634.8 1164.96  4655.6 1160.67  4776.9 1157.24  4785.3 1154.64
  4791.5 1154.98  4800.0 1133.26  4806.2 1129.26  4813.8 1117.90  4827.0 1117.40
  4871.0 1121.31  4921.2 1118.98  4927.4 1119.76  4955.4 1115.48  4955.9 1114.98
  4970.4 1115.48  4992.3 1116.58  4996.5 1119.16  5002.1 1119.16  5009.6 1123.18
  5029.6 1130.06  5049.6 1141.15  5069.6 1144.77  5109.6 1148.46  5199.6 1151.31
#Mann=4,-1,0
  4551.0    0.07       0  4571.9    0.12       0  4955.4    0.05       0
  4970.4    0.12       0
Bank Sta=4955.4,4970.4
Exp/Cntr=0.3,0.1

Type RM Length L Ch R = 1,6491,463,463,463
BEGIN DESCRIPTION:
SWEDE CREEK 14.0
END DESCRIPTION:
XS GIS Cut Line= 3
      2101060.86     13863752.40      2101125.00     13863475.00
      2101095.58     13863040.61
#Sta/Elev= 30
  4714.9 1147.60  4751.8 1147.53  4773.8 1146.32  4784.1 1147.13  4847.5 1142.66
  4855.9 1140.52  4866.2 1133.74  4885.1 1127.08  4890.2 1127.43  4897.0 1123.61
  4917.5 1117.26  4930.6 1115.67  4931.1 1115.17  4945.6 1115.67  5009.6 1115.73
  5019.7 1116.22  5029.7 1118.77  5049.7 1119.30  5079.8 1118.56  5099.8 1119.61
  5129.9 1124.52  5139.9 1127.99  5150.0 1130.29  5160.0 1134.61  5180.0 1139.92
  5240.2 1147.50  5320.3 1150.34  5340.4 1150.14  5372.5 1151.23  5435.0 1150.71
#Mann=3,-1,0
  4714.9    0.12       0  4930.6    0.05       0  4945.6    0.12       0
Bank Sta=4930.6,4945.6
Exp/Cntr=0.3,0.1

Type RM Length L Ch R = 1,6028,479,479,479
BEGIN DESCRIPTION:
SWEDE CREEK 13.0
END DESCRIPTION:
XS GIS Cut Line= 3
      2101151.13     13863766.30      2101525.00     13863575.00
      2101881.92     13863475.15
#Sta/Elev= 30
  4579.7 1144.08  4619.4 1142.12  4636.0 1139.26  4686.1 1135.95  4702.7 1132.52
  4747.1 1129.65  4769.3 1125.56  4775.0 1122.79  4785.9 1121.71  4833.2 1120.60
  4935.8 1117.31  4989.2 1114.84  4989.7 1114.34  5004.6 1114.84  5056.1 1117.05
  5062.0 1118.21  5072.4 1122.98  5090.2 1133.45  5095.4 1141.45  5103.5 1156.32
  5113.9 1158.07  5145.0 1159.76  5163.7 1163.08  5168.9 1162.60  5197.0 1168.44
  5237.1 1179.54  5248.9 1181.24  5315.8 1184.07  5332.0 1182.89  5370.3 1183.40
#Mann=5,-1,0
  4579.7    0.12       0  4833.2   0.035       0  4935.8    0.12       0
  4989.2    0.05       0  5004.6    0.12       0
Bank Sta=4989.2,5004.6
Exp/Cntr=0.3,0.1

Type RM Length L Ch R = 1,5549,444,444,444
BEGIN DESCRIPTION:
SWEDE CREEK 12.0
END DESCRIPTION:
XS GIS Cut Line= 3
      2101175.01     13863875.00      2101425.00     13863975.00
      2101921.03     13863995.43
#Sta/Elev= 30
  4731.0 1140.96  4740.4 1140.92  4752.5 1139.11  4784.8 1131.63  4794.3 1130.64
  4799.7 1131.00  4806.4 1129.38  4829.3 1121.18  4833.5 1120.64  4871.0 1118.20
  4929.5 1119.18  4967.9 1120.00  4985.4 1118.42  4997.6 1115.24  5002.6 1115.01
  5003.1 1114.51  5018.0 1115.01  5110.3 1115.76  5118.6 1126.80  5123.6 1141.14
  5130.4 1153.77  5140.4 1156.32  5160.4 1158.25  5210.4 1160.14  5250.5 1163.24
  5280.5 1167.93  5300.5 1173.11  5340.5 1175.69  5370.6 1178.85  5496.7 1180.26
#Mann=5,-1,0
  4731.0    0.12       0  4833.5   0.035       0  4929.5    0.12       0
  5002.6    0.05       0  5018.0    0.12       0
Bank Sta=5002.6,5018
Exp/Cntr=0.3,0.1

Type RM Length L Ch R = 1,5105,457,457,457
BEGIN DESCRIPTION:
SWEDE CREEK 11.0
END DESCRIPTION:
XS GIS Cut Line= 3
      2101024.99     13864074.99      2101175.00     13864325.00
      2101501.81     13864519.76
#Sta/Elev= 30
  4708.4 1143.54  4731.7 1143.48  4743.4 1138.34  4753.1 1136.62  4759.0 1132.85
  4766.7 1130.32  4774.5 1128.64  4801.7 1117.10  4825.0 1116.88  4849.5 1118.53
  4869.7 1119.67  4891.1 1115.44  4918.3 1115.31  5005.9 1114.82  5006.4 1114.32
  5020.8 1114.32  5021.3 1114.82  5029.2 1115.06  5044.8 1117.57  5050.6 1119.17
  5066.2 1119.56  5072.0 1123.05  5081.5 1125.54  5087.6 1130.54  5103.2 1140.47
  5130.4 1147.12  5161.6 1150.88  5206.9 1154.07  5327.0 1160.04  5380.4 1164.13
#Mann=6,-1,0
  4708.4    0.12       0  4849.5   0.035       0  4918.3    0.12       0
  5005.9    0.05       0  5021.3    0.12       0  5206.9   0.035       0
Bank Sta=5005.9,5021.3
Exp/Cntr=0.3,0.1

Type RM Length L Ch R = 1,4648,413,413,413
BEGIN DESCRIPTION:
SWEDE CREEK 10.0
END DESCRIPTION:
XS GIS Cut Line= 3
      2100501.79     13864262.80      2100775.00     13864475.00
      2101250.16     13864709.92
#Sta/Elev= 30
  4649.9 1153.08  4661.0 1152.48  4681.8 1148.52  4696.3 1147.09  4889.0 1139.77
  4938.8 1134.73  4945.2 1132.98  4953.3 1119.31  4959.6 1117.22  4982.3 1105.70
  4992.7 1103.82  5002.1 1103.56  5002.6 1103.06  5017.6 1103.56  5026.7 1105.01
  5032.3 1107.19  5049.1 1109.26  5071.6 1110.11  5087.8 1111.88  5241.3 1116.53
  5256.7 1119.15  5304.4 1134.24  5318.4 1140.97  5330.5 1145.12  5340.8 1146.96
  5352.8 1148.96  5385.7 1151.62  5412.6 1152.71  5453.0 1155.32  5525.9 1158.87
#Mann=7,-1,0
  4649.9    0.12       0  5002.1    0.05       0  5017.6    0.12       0
  5087.8   0.035       0  5304.4    0.12       0  5412.6    0.07       0
  5453.0   0.035       0
Bank Sta=5002.1,5017.6
Exp/Cntr=0.3,0.1

Type RM Length L Ch R = 1,4235,453,453,453
BEGIN DESCRIPTION:
SWEDE CREEK 9.0
END DESCRIPTION:
XS GIS Cut Line= 3
      2099845.55     13864436.43      2100525.00     13864775.00
      2101074.74     13864873.94
#Sta/Elev= 30
  4236.8 1184.06  4265.7 1174.80  4280.9 1171.82  4325.6 1167.19  4571.4 1151.05
  4660.7 1141.48  4802.9 1132.08  4853.2 1125.96  4870.0 1126.00  4875.6 1122.95
  4892.4 1123.62  4914.8 1128.01  4937.2 1127.49  4965.1 1124.04  4993.1 1108.40
  4998.5 1108.40  5008.5 1101.99  5009.0 1101.49  5024.0 1101.99  5046.7 1104.60
  5056.9 1108.43  5076.4 1112.27  5095.8 1113.40  5280.4 1113.98  5300.8 1116.01
  5311.2 1122.61  5323.8 1125.16  5402.4 1138.42  5472.1 1145.99  5554.5 1149.90
#Mann=5,-1,0
  4236.8    0.12       0  5008.5    0.05       0  5024.0    0.12       0
  5095.8   0.035       0  5323.8    0.12       0
Bank Sta=5008.5,5024
Exp/Cntr=0.3,0.1

Type RM Length L Ch R = 1,3782,445,445,445
BEGIN DESCRIPTION:
SWEDE CREEK 8.0
END DESCRIPTION:
XS GIS Cut Line= 3
      2099987.94     13865419.08      2100475.00     13865175.00
      2101077.61     13864929.74
#Sta/Elev= 30
  4451.3 1190.14  4473.8 1187.48  4490.5 1187.83  4540.8 1184.65  4638.2 1183.26
  4652.5 1181.34  4714.0 1178.75  4758.7 1171.72  4808.9 1159.08  4929.0 1150.90
  4937.4 1142.78  4943.0 1110.89  4959.8 1103.89  4982.1 1098.30  4996.1 1098.20
  4997.3 1096.89  4997.8 1096.39  5013.5 1096.89  5017.7 1101.93  5028.5 1106.50
  5058.9 1107.94  5082.5 1112.49  5125.9 1112.86  5212.0 1112.12  5297.1 1114.17
  5363.2 1121.98  5465.3 1127.31  5525.1 1133.39  5579.1 1142.37  5646.7 1148.49
#Mann=5,-1,0
  4451.3    0.12       0  4997.3    0.05       0  5013.5    0.12       0
  5125.9   0.035       0  5465.3    0.12       0
Bank Sta=4997.3,5013.5
Exp/Cntr=0.3,0.1

Type RM Length L Ch R = 1,3337,498,498,498
BEGIN DESCRIPTION:
SWEDE CREEK 7.0
END DESCRIPTION:
XS GIS Cut Line= 3
      2100675.01     13865574.99      2100825.00     13865425.00
      2101174.98     13865025.02
#Sta/Elev= 30
  4788.5 1155.36  4915.8 1146.18  4929.9 1143.94  4944.1 1129.84  4958.2 1113.06
  4972.3 1105.14  4999.6 1094.94  5000.1 1094.44  5015.8 1094.94  5028.6 1096.55
  5036.2 1100.43  5042.9 1100.98  5050.4 1104.27  5064.7 1106.00  5085.6 1105.50
  5099.8 1110.35  5114.0 1111.88  5218.2 1113.88  5317.8 1113.55  5361.8 1113.55
  5390.2 1116.27  5397.8 1119.99  5404.5 1120.64  5412.1 1126.97  5418.7 1129.69
  5425.8 1138.82  5439.6 1141.62  5461.4 1143.96  5468.1 1146.07  5532.1 1151.87
#Mann=5,-1,0
  4788.5    0.12       0  4999.6    0.05       0  5015.8    0.12       0
  5218.2   0.035       0  5317.8    0.12       0
Bank Sta=4999.6,5015.8
Exp/Cntr=0.3,0.1

Type RM Length L Ch R = 1,2839,466,466,466
BEGIN DESCRIPTION:
SWEDE CREEK 6.0
END DESCRIPTION:
XS GIS Cut Line= 3
      2100825.00     13865975.00      2101325.00     13865425.00
      2101375.01     13865224.97
#Sta/Elev= 30
  4260.7 1182.19  4296.2 1176.88  4359.7 1160.32  4402.3 1154.82  4494.2 1148.16
  4530.0 1143.52  4558.0 1137.03  4593.5 1131.28  4628.6 1122.16  4636.1 1122.30
  4642.8 1118.93  4696.4 1114.28  4848.3 1111.29  4940.2 1107.96  4946.2 1106.28
  4954.3 1106.05  4976.0 1096.99  4990.2 1093.11  5004.0 1092.94  5006.2 1091.23
  5006.7 1090.73  5022.4 1091.23  5063.3 1111.05  5068.4 1109.78  5076.2 1112.51
  5104.5 1116.98  5117.4 1129.85  5127.7 1137.68  5150.9 1143.06  5210.2 1148.23
#Mann=5,-1,0
  4260.7    0.12       0  4696.4   0.035       0  4946.2    0.12       0
  5006.2    0.05       0  5022.4    0.12       0
Bank Sta=5006.2,5022.4
Exp/Cntr=0.3,0.1

Type RM Length L Ch R = 1,2373,471,471,471
BEGIN DESCRIPTION:
SWEDE CREEK 5.0
END DESCRIPTION:
XS GIS Cut Line= 3
      2100876.87     13866078.78      2101525.00     13865825.00
      2101758.76     13865398.27
#Sta/Elev= 30
  4297.8 1181.10  4322.3 1178.42  4376.5 1162.41  4424.7 1154.31  4553.5 1144.88
  4599.0 1138.01  4623.5 1124.96  4628.8 1124.67  4647.9 1115.45  4677.7 1113.41
  4683.1 1127.76  4702.2 1126.25  4707.6 1113.73  4759.9 1113.27  4882.9 1112.26
  4918.7 1112.08  4940.1 1109.57  4954.5 1105.93  4974.2 1095.44  4983.0 1088.79
  4983.5 1088.29  4999.3 1088.79  5016.6 1091.56  5029.4 1098.39  5061.6 1106.43
  5073.7 1112.08  5127.1 1121.02  5176.4 1121.72  5199.1 1124.62  5480.4 1138.64
#Mann=6,-1,0
  4297.8    0.12       0  4759.9    0.07       0  4882.9   0.035       0
  4974.2    0.12       0  4983.0    0.05       0  4999.3    0.12       0
Bank Sta=4983,4999.3
Exp/Cntr=0.3,0.1

Type RM Length L Ch R = 1,1902,466,466,466
BEGIN DESCRIPTION:
SWEDE CREEK 4.0
END DESCRIPTION:
XS GIS Cut Line= 3
      2101525.00     13866225.00      2101725.00     13866225.00
      2102011.13     13866387.19
#Sta/Elev= 30
  4800.0 1115.13  4864.1 1115.42  4890.0 1114.35  4941.1 1093.86  4950.0 1089.23
  4960.0 1086.90  4970.0 1087.40  4971.0 1085.63  4971.5 1085.13  4989.1 1085.63
  4997.5 1091.60  5002.9 1091.60  5007.9 1100.51  5013.7 1100.32  5029.6 1111.99
  5035.3 1110.68  5045.5 1114.44  5051.2 1113.75  5057.5 1116.23  5067.1 1117.12
  5110.4 1115.35  5147.9 1115.77  5169.5 1119.21  5175.3 1121.17  5196.9 1125.53
  5218.5 1127.78  5241.4 1128.35  5264.4 1130.66  5287.4 1134.40  5328.9 1136.47
#Mann=5,-1,0
  4800.0    0.07       0  4864.1   0.035       0  4941.1    0.12       0
  4971.0    0.05       0  4989.1    0.12       0
Bank Sta=4971,4989.1
Exp/Cntr=0.3,0.1

Type RM Length L Ch R = 1,1436,460,460,460
BEGIN DESCRIPTION:
SWEDE CREEK 3.0
END DESCRIPTION:
XS GIS Cut Line= 3
      2101525.00     13866874.99      2101675.00     13866675.00
      2101984.48     13866641.30
#Sta/Elev= 30
  4746.1 1132.13  4768.0 1130.86  4782.6 1128.60  4788.8 1126.75  4796.1 1120.05
  4803.4 1118.39  4844.7 1117.31  4896.1 1118.60  4932.6 1117.92  4938.8 1116.30
  4959.6 1104.52  4968.0 1102.32  4974.2 1099.46  4980.7 1098.55  4988.8 1095.30
  4993.0 1092.56  4998.6 1092.56  5006.2 1087.76  5016.2 1085.72  5017.2 1083.81
  5017.7 1083.31  5035.3 1083.81  5041.8 1086.12  5056.4 1096.22  5066.5 1100.40
  5086.6 1104.63  5116.8 1108.87  5133.3 1114.07  5147.0 1116.31  5307.4 1117.83
#Mann=5,-1,0
  4746.1    0.12       0  4844.7   0.035       0  4980.7    0.12       0
  5017.2    0.05       0  5035.3    0.12       0
Bank Sta=5017.2,5035.3
Exp/Cntr=0.3,0.1

Type RM Length L Ch R = 1,976,474,474,474
BEGIN DESCRIPTION:
SWEDE CREEK 2.0
END DESCRIPTION:
XS GIS Cut Line= 3
      2101874.98     13867075.02      2102025.00     13866925.00
      2102025.00     13866724.96
#Sta/Elev= 30
  4788.3 1126.81  4802.5 1127.03  4830.7 1126.79  4844.9 1127.12  4887.3 1127.12
  4901.5 1126.58  4915.6 1125.63  4929.7 1119.00  4943.9 1108.44  4958.0 1100.75
  4972.2 1094.08  4986.3 1084.55  4996.9 1083.27  5000.5 1083.27  5001.4 1082.97
  5001.9 1082.47  5019.0 1082.47  5019.5 1082.97  5020.5 1084.77  5030.5 1091.18
  5040.5 1096.54  5070.5 1108.75  5080.5 1112.14  5100.5 1117.20  5110.5 1119.02
  5130.5 1119.62  5170.5 1119.05  5180.5 1119.22  5190.5 1118.68  5200.5 1118.54
#Mann=3,-1,0
  4788.3    0.12       0  5001.4    0.05       0  5019.5    0.12       0
Bank Sta=5001.4,5019.5
Exp/Cntr=0.3,0.1

Type RM Length L Ch R = 1,502,0,0,0
BEGIN DESCRIPTION:
SWEDE CREEK 1.0
END DESCRIPTION:
XS GIS Cut Line= 3
      2102425.00     13867025.00      2102425.00     13866825.00
      2102425.00     13866625.00
#Sta/Elev= 30
  4804.2 1114.60  4824.2 1117.65  4844.2 1118.27  4864.2 1116.99  4884.2 1104.38
  4894.2 1101.99  4904.2 1097.87  4924.2 1093.34  4934.2 1089.96  4964.2 1083.61
  4974.2 1080.15  4975.1 1078.12  4975.6 1077.62  4993.2 1078.12  4994.2 1083.28
  5001.7 1086.19  5006.7 1086.19  5014.2 1091.46  5024.2 1095.38  5034.2 1101.32
  5074.2 1117.40  5084.2 1119.77  5094.2 1120.50  5104.2 1133.78  5114.2 1141.20
  5124.2 1145.12  5144.2 1148.34  5164.2 1150.57  5194.2 1152.92  5204.2 1153.02
#Mann=3,-1,0
  4804.2    0.12       0  4975.1    0.05       0  4993.2    0.12       0
Bank Sta=4975.1,4993.2
Exp/Cntr=0.3,0.1

Chan Stop Cuts=-1
